HEC-RAS study Denton Creek.prj: Denton Creek Base Level Engineering

--- Denton Creek.g01 (geometry) --- (continued)

Type RM Length L Ch R = 1 ,533876  ,485,485,485
BEGIN DESCRIPTION:
Denton Creek 286.0
END DESCRIPTION:
XS GIS Cut Line= 3
       2193715.4      7261044.27       2193215.6      7260396.59
      2192828.99      7259659.98
#Sta/Elev= 30
  4052.1 1030.98  4266.5 1018.61  4287.4 1020.41  4337.2 1013.76  4407.6 1014.86
  4465.8 1012.52    4474 1015.62  4480.3 1012.51    4487 1016.13  4530.1 1011.09
  4579.9 1012.55  4644.3 1010.03  4673.3 1003.09  4714.9  1006.3  4752.1 1001.95
  4779.2 1006.03  4824.8 1003.38  4911.3  999.16  4983.1  1002.2  4990.6  999.03
  4991.7  995.02  4993.7  994.52  5007.2  995.02  5043.6 1002.55  5069.8  1001.4
  5172.8 1003.17  5358.5 1008.28  5510.1 1020.43  5627.7 1025.66  5702.1 1033.81
#Mann= 8 ,-1 , 0
  4052.1     .05       0  4407.6     .16       0  4824.8     .05       0
  4991.7    .035       0  5007.2     .05       0  5069.8     .16       0
  5172.8     .05       0  5358.5     .16       0
Bank Sta=4991.7,5007.2
XS Rating Curve= 0 ,0
Exp/Cntr=0.3,0.1

Type RM Length L Ch R = 1 ,533391  ,266,266,266
BEGIN DESCRIPTION:
Denton Creek 285.0
END DESCRIPTION:
XS GIS Cut Line= 3
      2194066.03      7260651.95        2193529.        7260110.
      2192928.99      7259609.99
#Sta/Elev= 30
  4240.1    1025    4296 1022.16  4324.3 1017.85  4409.1 1023.31  4472.7    1024
  4650.2 1015.74  4748.5 1011.28  4847.5 1004.31  4868.7 1000.71  4918.2  999.33
  4953.6 1004.46  4967.7  1000.2    4974   993.8    4976   993.3  4989.6   993.8
  5006.3  995.34  5016.7 1001.16  5024.5 1002.16  5059.7  999.84  5172.9  999.98
  5223.7 1000.95    5251 1005.86  5303.8 1005.48  5400.7 1007.47  5581.2 1017.82
  5641.6 1021.19  5649.4 1019.59  5670.2 1023.67  5741.8 1028.46  5784.1  1035.4
#Mann= 6 ,-1 , 0
  4240.1     .05       0  4650.2     .16       0    4974     .07       0
  4989.6     .16       0  5303.8     .05       0  5581.2     .16       0
Bank Sta=4974,4989.6
XS Rating Curve= 0 ,0
Exp/Cntr=0.3,0.1

Type RM Length L Ch R = 1 ,533125  ,137,137,137
BEGIN DESCRIPTION:
Denton Creek302
END DESCRIPTION:
XS GIS Cut Line= 3
      2194108.95      7260312.81      2193613.84      7259824.48
      2193193.84      7259399.23
#Sta/Elev= 30
  4458.8 1017.33  4637.6 1009.49  4651.7 1006.66  4658.7 1007.92  4672.9  1004.5
    4680 1008.66    4687 1006.49  4694.1 1008.41  4750.7 1006.34  4764.8 1007.49
  4814.3 1003.76  4906.3    1001  4962.8 1001.66  4998.2  996.72  5004.5  993.62
  5006.5  993.12  5020.1  993.62  5026.4  996.93  5068.9 1000.12  5111.3 1000.98
  5132.6  998.96  5167.9 1001.73  5245.6 1000.88  5343.2 1003.97  5415.3  1006.9
  5595.7 1020.46  5641.6 1022.64  5655.7 1026.91  5733.2 1033.16  5751.9 1035.05
#Mann= 7 ,-1 , 0
  4458.8     .16       0  5004.5     .07       0  5020.1     .16       0
  5343.2     .05       0  5595.7     .16       0  5655.7     .05       0
  5733.2     .16       0
Bank Sta=5004.5,5020.1
XS Rating Curve= 0 ,0
Exp/Cntr=0.3,0.1

Type RM Length L Ch R = 1 ,532988  ,463,463,463
BEGIN DESCRIPTION:
Denton Creek 284.0
END DESCRIPTION:
XS GIS Cut Line= 3
      2194208.41       7260181.9      2193943.25      7259972.26
      2193278.97      7259259.97
#Sta/Elev= 30
  4504.3 1020.22  4562.4 1016.47  4618.4 1014.47  4682.5 1008.86  4818.8 1003.42
  4841.8 1001.27  4917.6  999.17  4924.9 1000.53  4953.2  999.18  4974.2  999.61
  4981.6  999.11  4994.8  990.07  4996.8  989.57  5010.4  990.07  5016.8  994.47
  5030.9  999.53  5115.9  998.68  5122.8 1000.95  5130.1  998.83  5200.9  998.27
  5347.5 1004.61  5387.9 1005.83  5427.1 1007.46    5489 1013.23  5524.8 1015.47
  5630.4 1022.82  5661.7 1025.33  5771.9 1032.42  5798.6 1034.14  5816.3 1035.11
#Mann= 11 ,-1 , 0
  4504.3     .05       0  4994.8    .035       0  5010.4     .05       0
  5347.5    .063       0  5387.9     .05       0    5489    .063       0
  5524.8     .05       0  5630.4    .063       0  5661.7     .05       0
  5771.9    .063       0  5798.6     .05       0
Bank Sta=4994.8,5010.4
XS Rating Curve= 0 ,0
Exp/Cntr=0.3,0.1

Type RM Length L Ch R = 1 ,532525  ,623,623,623
BEGIN DESCRIPTION:
Denton Creek 283.0
END DESCRIPTION:
XS GIS Cut Line= 3
      2194500.64      7259851.51        2194179.        7259560.
      2193590.78      7258986.23
#Sta/Elev= 30
  4561.7 1019.35  4606.2 1018.45  4648.7  1014.5  4698.8 1012.89  4733.9 1009.59
  4797.4 1007.98  4811.6 1005.34  4896.8 1001.02  4925.2  996.96  4943.4  998.75
  4960.3  999.27  4968.1 1003.03  4981.9  994.52  4984.6   986.9  4986.6   986.4
  5000.3   986.9  5002.9  991.06  5031.1  997.74  5045.3  998.43    5116  996.87
  5158.5  997.84  5186.7     996  5229.2  996.52  5278.6  994.38  5342.3  998.54
  5490.8 1002.67  5512.1 1005.86  5582.6 1008.39  5674.7 1016.07  5817.5 1024.58
#Mann= 5 ,-1 , 0
  4561.7     .05       0  4943.4     .16       0  4968.1     .05       0
  4984.6    .035       0  5000.3     .05       0
Bank Sta=4984.6,5000.3
XS Rating Curve= 0 ,0
Exp/Cntr=0.3,0.1

Type RM Length L Ch R = 1 ,531902  ,701,701,701
BEGIN DESCRIPTION:
Denton Creek 282.0
END DESCRIPTION:
XS GIS Cut Line= 3
      2194748.15      7259285.29      2194540.96       7259069.1
      2193828.99      7258609.99
#Sta/Elev= 30
  4647.6 1019.84  4728.2 1015.83  4778.2 1014.76  4884.2 1007.78  4905.2 1005.32
  4919.4 1001.03  4926.6  996.58  4933.5  995.59  4940.8   998.6  4961.3  1000.1
  4970.1  996.26  4976.1  996.15  4985.1  990.64  4989.4  984.71  4991.4  984.21
  5005.1  984.71  5006.4  987.24  5011.5  985.33  5027.6  998.55  5033.5   996.7
  5048.7  998.28  5070.7  996.36  5136.5  993.92  5209.1  995.07  5230.2  992.75
  5302.8  997.63    5392  996.69  5490.2   998.1  5723.9  1006.2  5794.2  1009.8
#Mann= 8 ,-1 , 0
  4647.6     .05       0  4728.2     .16       0  4989.4     .07       0
  5005.1     .16       0  5011.5     .05       0  5070.7     .16       0
    5392     .05       0  5723.9     .16       0
Bank Sta=4989.4,5005.1
XS Rating Curve= 0 ,0
Exp/Cntr=0.3,0.1

Type RM Length L Ch R = 1 ,531201  ,1013,1013,1013
BEGIN DESCRIPTION:
Denton Creek 280.0
END DESCRIPTION:
XS GIS Cut Line= 3
      2195074.78       7259003.6        2194529.        7258360.
      2194009.94      7257915.56
#Sta/Elev= 30
  4143.5 1008.93  4249.7 1003.94  4606.3  998.53  4682.5  994.31  4793.5  993.64
  4845.4  993.47  4959.4  993.62  4973.7  989.94  4986.5  980.11  4988.5  979.61
  5002.4  980.11  5008.8  983.37  5015.3  982.53  5037.3  987.75  5043.9  992.44
  5086.7  991.99    5131  995.03  5193.2  995.53  5207.4  998.04  5232.5  996.12
  5256.8  997.11  5264.7  999.92  5313.9 1003.86  5334.8 1001.54  5363.3 1006.34
  5412.7 1007.35  5420.4  1009.6  5568.6 1018.86  5582.8 1021.99  5670.7 1026.49
#Mann= 9 ,-1 , 0
  4143.5     .05       0  4606.3     .16       0  4793.5     .05       0
  4845.4     .16       0  4986.5     .07       0  5002.4     .16       0
    5131     .05       0  5232.5     .16       0  5264.7     .05       0
Bank Sta=4986.5,5002.4
XS Rating Curve= 0 ,0
Exp/Cntr=0.3,0.1

Type RM Length L Ch R = 1 ,530188  ,862,862,862
BEGIN DESCRIPTION:
Denton Creek 278.0
END DESCRIPTION:
XS GIS Cut Line= 3
      2195728.99      7258409.99      2195204.93      7257820.09
      2194849.92      7257187.23
#Sta/Elev= 30
  4129.7 1014.97  4228.8 1009.51  4441.2  992.72  4576.5  988.08  4696.2  991.42
  4802.4  988.55    4966   990.6  4976.2  990.07    4982  986.99  4989.9  975.74
  4991.9  975.24  5005.9  975.74  5025.3  988.84  5246.7  1000.6  5311.7 1000.21
  5327.7 1002.69  5333.4 1000.13  5349.4 1002.19  5355.1  999.02  5361.8 1000.44
  5371.1  999.58  5392.7 1003.91  5400.4 1009.74  5408.7 1012.38  5473.8 1017.66
  5503.6    1023  5517.1 1022.97  5538.8 1018.72  5614.1 1018.55  5644.4 1020.86
#Mann= 5 ,-1 , 0
  4129.7     .05       0  4576.5     .16       0  4989.9     .07       0
  5005.9     .16       0  5361.8     .05       0
Bank Sta=4989.9,5005.9
XS Rating Curve= 0 ,0
Exp/Cntr=0.3,0.1

Type RM Length L Ch R = 1 ,529326  ,821,821,821
BEGIN DESCRIPTION:
Denton Creek 276.0
END DESCRIPTION:
XS GIS Cut Line= 3
        2196029.      7258010.03        2195929.        7257410.
        2195629.        7256910.
#Sta/Elev= 30
    4384 1003.11  4465.1  996.98  4566.5  992.65  4607.1  989.16  4667.9  986.26
  4717.9  986.23  4728.7  984.84    4749   986.4  4890.9  984.71  4964.4  987.21
  4982.2  986.58  4989.8  979.69  4995.2  979.69  4997.9  975.66  4999.9  975.16
  5013.9  975.66    5037     984  5042.8  984.06  5050.6  986.95  5101.1  985.65
  5116.7  986.55  5122.5  985.31  5143.9  986.48  5190.6  985.34  5307.2  990.04
  5365.5  995.28  5392.7  998.91    5451 1003.28  5552.1 1020.37  5575.4 1021.72
#Mann= 4 ,-1 , 0
    4384     .05       0  4717.9     .16       0  4997.9     .07       0
  5013.9     .16       0
Bank Sta=4997.9,5013.9
XS Rating Curve= 0 ,0
Exp/Cntr=0.3,0.1

Type RM Length L Ch R = 1 ,528505  ,567,567,567
BEGIN DESCRIPTION:
Denton Creek 274.0
END DESCRIPTION:
XS GIS Cut Line= 3
        2196379.      7258060.01        2196679.        7257460.
        2196579.        7256860.
#Sta/Elev= 30
  4290.8 1004.79  4349.5 1002.15  4366.3  999.68  4388.6  998.17  4416.6  997.69
  4528.4  988.21  4679.5  984.51  4827.5  984.64  4902.9  983.19  4908.5  983.98
  4930.9  982.35  4953.2  983.42  4958.8  980.11  4964.2  980.11  4971.8  975.25
  4981.4  971.85  4983.4  971.35  4997.6  971.85  5022.5  982.99  5042.7  985.75
  5111.2   983.6  5144.1  983.81  5232.8   989.2  5316.5  992.52  5377.3  993.39
  5415.3  997.44  5420.4  996.67  5438.1   997.7    5542 1007.24  5569.9 1008.47
#Mann= 4 ,-1 , 0
  4290.8     .05       0  4679.5     .16       0  4981.4     .07       0
  4997.6     .16       0
Bank Sta=4981.4,4997.6
XS Rating Curve= 0 ,0
Exp/Cntr=0.3,0.1

Type RM Length L Ch R = 1 ,527938  ,517,517,517
BEGIN DESCRIPTION:
Denton Creek 273.0
END DESCRIPTION:
XS GIS Cut Line= 3
      2198021.01      7258041.03      2197280.81      7257779.46
      2196978.99      7256859.98
#Sta/Elev= 30
  3749.8 1017.93  3798.8 1017.18  3868.6 1012.03    3979 1014.24  4009.9 1012.77
  4027.7 1011.49  4040.8 1008.25  4059.5 1000.72  4104.3 1000.72  4112.5  999.51
  4128.2 1003.66  4197.4  999.14  4523.9  986.42    4608  984.56  4850.3  985.93
  4892.1  980.22  4934.2  980.47  4955.3  976.59  4965.8     977  4984.9  970.65
  4987.4  970.15  5009.9  970.65  5018.4  980.08  5035.9  983.26  5099.6  983.93
  5186.8  981.46  5258.7  984.11    5423  997.73    5471 1005.03  5502.6 1007.22
#Mann= 5 ,-1 , 0
  3749.8     .16       0  4104.3     .05       0  4523.9     .16       0
  4984.9     .07       0  5009.9     .16       0
Bank Sta=4984.9,5009.9
XS Rating Curve= 0 ,0
Exp/Cntr=0.3,0.1

Type RM Length L Ch R = 1 ,527421  ,1054,1054,1054
BEGIN DESCRIPTION:
Denton Creek 272.0
END DESCRIPTION:
XS GIS Cut Line= 3
      2198029.03      7257360.02        2197529.        7257010.
      2197028.98      7256809.99
#Sta/Elev= 30
  4385.3 1011.14    4422 1002.12  4479.1  994.52  4592.8  985.25  4693.5  981.03
  4775.4  981.67  4824.3  983.16  4851.4  982.15  4952.5   983.7  4967.3  982.29
  4982.1  978.68  4988.2  974.62  4992.6   970.1    4998  969.77  5000.5  969.27
    5023  969.77    5028  976.37  5040.1  981.98  5058.9  984.54  5064.3  983.48
  5146.3  981.22  5157.2  979.17  5166.6  979.48  5178.8  982.42  5196.3  980.46
  5302.2  987.08  5394.2  995.06  5435.9  997.45  5519.4 1006.81  5534.2 1006.93
#Mann= 6 ,-1 , 0
  4385.3     .05       0  4775.4     .16       0    4998     .07       0
    5023     .16       0  5146.3     .05       0  5302.2     .16       0
Bank Sta=4998,5023
XS Rating Curve= 0 ,0
Exp/Cntr=0.3,0.1

Type RM Length L Ch R = 1 ,526367  ,531,531,531
BEGIN DESCRIPTION:
Denton Creek 270.0
END DESCRIPTION:
XS GIS Cut Line= 3
      2198838.21       7256474.6        2197979.        7256210.
      2197049.45      7256073.87
#Sta/Elev= 30
  4121.4 1012.67  4235.7 1005.32  4499.6   993.1  4525.6   992.4  4661.6  983.61
  4748.4  979.59  4905.6  980.89  4971.4  979.35    4989  973.06  4997.5  968.07
    5000  967.57  5022.5  968.07    5023  970.82    5040  978.69  5055.4  980.54
  5182.1  978.34  5242.8  979.97  5283.2  978.25  5343.8  977.41  5399.7  979.11
  5515.7  979.24    5647  982.29  5707.7  984.69  5808.8  993.61  5849.2  995.23
  5878.8  999.53  5909.8 1000.91  5919.9 1000.08    5930 1002.06  5959.9  1004.2
#Mann= 6 ,-1 , 0
  4121.4     .16       0  4499.6     .05       0  4905.6     .16       0
  4997.5     .07       0  5022.5     .16       0    5040     .05       0
Bank Sta=4997.5,5022.5
XS Rating Curve= 0 ,0
Exp/Cntr=0.3,0.1

Type RM Length L Ch R = 1 ,525836  ,477,477,477
BEGIN DESCRIPTION:
Denton Creek 269.0
END DESCRIPTION:
XS GIS Cut Line= 4
      2198729.02      7256260.01        2198079.        7255710.
      2197483.13      7255432.81      2196733.24      7255808.03
#Sta/Elev= 30
  4136.5  1009.8  4164.5 1009.13  4215.1 1000.14  4242.5  999.86    4274  996.78
  4371.1  987.55  4512.8  980.06  4619.4  977.32  4894.8  979.55  4952.3  979.15
  4973.3  974.43  4980.8  973.96  4989.7  968.17  4992.2  967.67  5014.7  968.17
    5048  972.84  5070.8   973.6  5093.7  977.05  5099.2  979.73  5131.4  980.52
  5208.1  978.59  5213.7  980.32  5230.6  978.55  5242.1  980.17  6027.2  981.41
  6384.9   991.8  6457.5  997.01  6474.3  994.02  6479.9  994.97  6483.7  993.12
#Mann= 6 ,-1 , 0
  4136.5     .16       0    4274     .05       0  4894.8     .16       0
  4973.3     .05       0  4989.7    .035       0  5014.7     .05       0
Bank Sta=4989.7,5014.7
XS Rating Curve= 0 ,0
Exp/Cntr=0.3,0.1

Type RM Length L Ch R = 1 ,525359  ,587,587,587
BEGIN DESCRIPTION:
Denton Creek 268.0
END DESCRIPTION:
XS GIS Cut Line= 3
      2198788.33      7256155.64      2198215.85       7255133.3
      2197316.61       7254399.6
#Sta/Elev= 30
    4067 1002.07  4141.1  997.78  4245.4  990.66  4607.2  976.91  4703.8  975.44
    4791  977.92  4953.1   977.6  4980.5  973.96  4989.7  967.36  4992.2  966.86
  5014.7  967.36  5024.7  972.29  5047.7  978.39    5079  977.69  5223.7  977.39
  5237.7  975.03  5292.1  976.35  5299.5  976.51  5415.1  977.46  5451.4  977.45
  5899.9  978.31  6041.6  982.18  6097.4  984.59  6155.5  987.08  6184.2  991.24
  6268.9  995.53  6347.2 1003.43  6355.1  1006.2  6361.5 1004.25  6399.3 1003.98
#Mann= 11 ,-1 , 0
    4067     .16       0  4141.1     .05       0  4989.7    .035       0
  5014.7     .05       0    5079     .05       0  5292.1     .05       0
  5299.5     .05       0  5415.1     .05       0  5451.4     .05       0
  6041.6     .05       0  6097.4     .16       0
Bank Sta=4989.7,5014.7
XS Rating Curve= 0 ,0
Exp/Cntr=0.3,0.1

Type RM Length L Ch R = 1 ,524772  ,482,482,482
BEGIN DESCRIPTION:
Denton Creek 267.0
END DESCRIPTION:
XS GIS Cut Line= 4
      2199240.64      7256145.03        2198879.        7255160.
      2198687.47      7254738.62      2198642.06      7253917.26
#Sta/Elev= 30
  3936.8 1020.38  3963.5 1020.09  4048.7 1029.33  4101.7 1021.27  4134.7 1011.94
    4185 1004.31    4336  993.94  4406.1  988.94  4549.4  979.78  4651.5  976.28
  4737.6  974.33  4841.3   974.7  4931.7  976.43  4954.2  977.18  4976.2  974.72
  4983.5  971.09  4988.9  971.09  4994.9  967.62  4995.6   965.5  4998.1     965
  5020.6   965.5    5041  976.37  5242.1  974.33  5434.2  990.91  5507.2  992.85
    5688 1003.09  5798.1  1001.8  6068.6 1007.51  6108.6 1005.58  6271.6 1008.67
#Mann= 9 ,-1 , 0
  3936.8     .16       0  4101.7     .05       0    4336     .05       0
  4406.1     .05       0  4841.3     .05       0  4931.7     .05       0
  4995.6    .035       0  5020.6     .05       0  5434.2     .05       0
Bank Sta=4995.6,5020.6
XS Rating Curve= 0 ,0
Exp/Cntr=0.3,0.1

Type RM Length L Ch R = 1 ,524290  ,474,474,474
BEGIN DESCRIPTION:
Denton Creek 266.0
END DESCRIPTION:
XS GIS Cut Line= 3
        2199679.        7255710.        2199279.        7254910.
        2199229.      7254510.04
#Sta/Elev= 30
  4116.7 1027.33  4181.1 1018.38  4206.1 1012.91  4236.9 1008.79  4384.4  994.86
    4399   994.4  4438.1  987.84  4474.5  984.05  4608.6  973.92  4675.7  971.87
  4801.5  972.96  4840.6  975.15  4921.7   976.4    4944  976.09    4979  971.09
  4988.8  969.31  4995.8  964.74  4998.3  964.24  5020.8  964.74  5021.2  966.22
  5041.4  974.65  5059.3  973.94    5122  972.62  5191.1  974.83  5215.2  977.29
  5222.8   979.6    5290  984.16  5303.4   986.7  5333.6  987.44  5414.2  994.42
#Mann= 9 ,-1 , 0
  4116.7     .16       0  4181.1     .05       0  4384.4     .05       0
    4979     .05       0  4995.8    .035       0  5020.8     .05       0
  5059.3     .05       0  5191.1     .05       0    5290     .16       0
Bank Sta=4995.8,5020.8
XS Rating Curve= 0 ,0
Exp/Cntr=0.3,0.1

Type RM Length L Ch R = 1 ,523816  ,750,750,750
BEGIN DESCRIPTION:
Denton Creek 265.0
END DESCRIPTION:
XS GIS Cut Line= 3
      2199945.05      7255750.08      2199663.86      7254544.58
      2199528.98      7254359.97
#Sta/Elev= 30
  3957.5 1012.62  3978.1 1011.77    4005 1004.33  4010.1 1007.52  4029.5  1006.9
  4052.7 1012.39  4067.9 1013.01  4101.3 1005.62  4318.2  992.13  4368.3  985.16
  4398.2  983.22  4403.3  980.92  4603.4   972.8  4645.6  971.42  4706.3  973.72
  4748.3  972.52  4820.1  973.96  4839.1  976.02  4869.5  974.08  4922.8   975.6
  4953.6  972.52  4970.7   973.3  4984.4  971.45  4992.5  963.51    4995  963.01
  5017.5  963.51  5025.5  975.17  5087.1  974.06  5144.9   977.7    5424   998.7
#Mann= 8 ,-1 , 0
  3957.5     .16       0  4067.9     .05       0  4603.4     .16       0
  4869.5     .05       0  4970.7     .16       0  4992.5     .07       0
  5017.5     .16       0  5144.9     .05       0
Bank Sta=4992.5,5017.5
XS Rating Curve= 0 ,0
Exp/Cntr=0.3,0.1

Type RM Length L Ch R = 1 ,523066  ,874,874,874
BEGIN DESCRIPTION:
Denton Creek301
END DESCRIPTION:
XS GIS Cut Line= 4
      2201202.86      7256200.74      2200798.45      7255003.02
      2200143.33       7254392.2      2199513.87      7254257.81
#Sta/Elev= 30
  3172.1  1009.9  3288.6  996.96  3477.4  984.31  3729.1  983.39  4270.2  977.77
  4692.9  972.96  4721.2  975.69  4735.4  975.36  4749.5  972.35  4784.7   972.1
  4805.7  974.14  4827.2  971.25  4883.9  972.31  4898.1  975.96  4919.1  972.53
  4961.6  974.23  4968.7  973.11  4975.7  971.08  4984.2  962.31  4986.7  961.81
  5009.2  962.31  5010.9   967.7  5016.4  969.43  5039.2  971.79  5081.8   972.8
  5463.2  972.07  5601.5  979.51  5656.1  980.29  5700.5  984.18  5975.6  999.64
#Mann= 5 ,-1 , 0
  3172.1     .05       0  4270.2     .16       0  4984.2     .07       0
  5009.2     .16       0  5016.4     .05       0
Bank Sta=4984.2,5009.2
XS Rating Curve= 0 ,0
Exp/Cntr=0.3,0.1

Type RM Length L Ch R = 1 ,522192  ,561,561,561
BEGIN DESCRIPTION:
Denton Creek 263.0
END DESCRIPTION:
XS GIS Cut Line= 3
      2201178.97      7253460.02        2200479.        7253860.
      2199328.98      7254210.01
#Sta/Elev= 30
  4220.6  1017.2  4293.3    1013  4309.1 1008.27    4316 1008.73  4330.7 1004.19
  4373.9  999.52  4389.7  994.19  4411.3  990.59  4513.5  982.54    4610  977.73
  4712.2  968.59    4718  966.69  4749.7  970.07    4777   968.7  4901.8  970.59
  4938.3  972.31  4954.1  968.58    4979  966.91  4991.3  960.88  4993.8  960.38
  5016.3  960.88  5018.9  968.56  5037.2  972.19    5194  968.98  5698.8  973.28
  5998.9  991.74  6051.2  997.46  6103.4  999.19  6134.8 1002.45  6228.9 1004.87
#Mann= 6 ,-1 , 0
  4220.6     .16       0    4316     .05       0  4901.8     .16       0
    4979     .05       0  4991.3    .035       0  5016.3     .05       0
Bank Sta=4991.3,5016.3
XS Rating Curve= 0 ,0
Exp/Cntr=0.3,0.1

Type RM Length L Ch R = 1 ,521631  ,1073,1073,1073
BEGIN DESCRIPTION:
Denton Creek 262.0
END DESCRIPTION:
XS GIS Cut Line= 3
        2201029.        7253360.        2200629.        7253360.
      2199329.02        7253110.
#Sta/Elev= 30
  4552.5 1004.97  4592.5 1003.73    4616 1001.19  4662.5  998.07  4682.5  994.03
  4712.5  983.83  4732.5  980.33  4862.5   975.8  4892.5  971.28  4902.5  967.69
  4932.5  963.59  4962.7   965.4  4978.5  962.33  4980.7  957.95  4983.2  957.45
  5005.7  957.95  5013.6  960.73  5064.5  963.01  5082.3  967.68  5115.4  969.51
  5359.8  967.19  5404.1  967.58  5410.7  968.87  5441.3  966.24  5461.7  968.46
  5573.7  967.43  5685.7   969.8  5848.6  980.51  5960.6   989.9  6276.3  1003.1
#Mann= 4 ,-1 , 0
  4552.5     .16       0    4616     .05       0  4980.7    .035       0
  5005.7     .05       0
Bank Sta=4980.7,5005.7
XS Rating Curve= 0 ,0
Exp/Cntr=0.3,0.1

Type RM Length L Ch R = 1 ,520558  ,1213,1213,1213
BEGIN DESCRIPTION:
Denton Creek 260.0
END DESCRIPTION:
XS GIS Cut Line= 3
      2201429.03      7253110.03      2200580.76      7252040.36
      2200028.99        7252010.
#Sta/Elev= 30
  4240.7 1009.87  4312.1 1003.03  4382.5  989.92  4446.6  984.88  4454.7  982.55
  4475.5  982.85  4489.9  979.55  4510.7  981.86  4525.1  979.52  4539.6  981.54
    4554  980.03  4568.4  983.41  4581.5  982.41  4610.9   977.5    4711  970.91
  4839.2  964.83    4898  964.41  4959.4  966.53  4967.4  965.51  4975.7  956.72
  4978.2  956.22  5000.7  956.72  5044.8  966.14  5076.1  965.21  5609.3  964.62
  5777.9  977.63    5858  981.16  5908.1  986.95  6098.4  995.96  6158.5  996.09
#Mann= 6 ,-1 , 0
  4240.7     .16       0  4581.5     .05       0    4898     .16       0
  4975.7     .07       0  5000.7     .16       0  5076.1     .05       0
Bank Sta=4975.7,5000.7
XS Rating Curve= 0 ,0
Exp/Cntr=0.3,0.1

Type RM Length L Ch R = 1 ,519345  ,1171,1171,1171
BEGIN DESCRIPTION:
Denton Creek 259.0
END DESCRIPTION:
XS GIS Cut Line= 3
      2202529.03      7252460.03        2201729.        7251660.
      2200519.49       7250498.8
#Sta/Elev= 30
  3857.1 1003.74  3956.1  986.09  4026.8  978.53  4062.7  976.98  4097.6  973.61
  4196.5  969.46  4479.4  963.33  4733.5  960.98  4776.4  959.95  4918.5  962.29
  4960.2  962.84    4990   955.4  4992.5   954.9    5015   955.4  5016.7  958.96
  5023.9  962.59  5518.9  960.29  5996.9  964.25  6098.8   965.2  6120.2  959.91
  6148.5  965.13  6211.1  963.49  6268.6  963.72  6332.4  966.56    6417  974.01
  6445.3  978.93  6473.9  980.04  6568.7  985.18  6583.3  985.42  6665.2  988.31
#Mann= 11 ,-1 , 0
  3857.1     .16       0  4062.7     .05       0  4733.5     .16       0
  4918.5     .05       0    4990    .035       0    5015     .05       0
  5996.9     .16       0  6211.1     .05       0  6473.9     .16       0
  6568.7     .05       0  6583.3     .16       0
Bank Sta=4990,5015
XS Rating Curve= 0 ,0
Exp/Cntr=0.3,0.1

Type RM Length L Ch R = 1 ,518174  ,169,169,169
BEGIN DESCRIPTION:
Denton Creek300
END DESCRIPTION:
XS GIS Cut Line= 3
      2203098.23      7251738.38      2202170.08      7250787.83
      2201407.24      7250029.03
#Sta/Elev= 30
  4039.4  996.86  4220.2  985.65  4285.3  978.85  4398.4  974.78  4589.3  960.36
  4737.7  958.48    4766  965.62  4794.7  961.51  4837.2   958.8  4934.7  960.19
  4978.2  959.37  4992.3  954.42    4994  950.39  4996.5  949.89    5019  950.39
  5020.6  954.56  5027.8  959.35  5074.8  960.24  5678.3  957.67  5954.1  961.24
  5990.9  958.74  6003.6  961.42  6128.6  961.08  6317.1  971.17  6335.9  973.12
    6343  967.07    6350  964.94  6364.2  968.47  6371.2  974.22  6443.9  979.71
#Mann= 11 ,-1 , 0
  4039.4     .16       0  4220.2     .05       0  4794.7     .16       0
  4837.2     .05       0  4934.7     .16       0    4994     .07       0
    5019     .16       0  5074.8     .05       0  5990.9     .16       0
  6128.6     .05       0  6317.1     .16       0
Bank Sta=4994,5019
XS Rating Curve= 0 ,0
Exp/Cntr=0.3,0.1

Type RM Length L Ch R = 1 ,518005  ,803,803,803
BEGIN DESCRIPTION:
Denton Creek 256.0
END DESCRIPTION:
XS GIS Cut Line= 3
      2203222.15      7251644.06      2202696.93      7251103.38
      2201588.92      7249961.05
#Sta/Elev= 30
  4072.5  990.73  4084.7  991.56    4106  989.51    4113  991.47  4155.4  985.02
  4501.9  966.48  4615.1  958.66  4749.3  957.63  4968.7  959.66  4989.8  951.52
  4991.5  949.72    4994  949.22  5016.5  949.72  5018.1  954.44  5025.3  958.99
  5060.6  961.04  5117.2  958.81  5562.7  957.48  5859.8  958.11    5895  961.43
  5916.4  957.78  5923.3  961.42  5930.5  960.09    5973  959.44  6029.3  959.98
  6043.5  961.68  6057.6  959.78  6071.8  960.02  6227.4  966.52  6417.7  976.78
#Mann= 3 ,-1 , 0
  4072.5     .05       0  4991.5    .035       0  5016.5     .05       0
Bank Sta=4991.5,5016.5
XS Rating Curve= 0 ,0
Exp/Cntr=0.3,0.1

Type RM Length L Ch R = 1 ,517202  ,508,508,508
BEGIN DESCRIPTION:
Denton Creek 255.0
END DESCRIPTION:
XS GIS Cut Line= 3
      2204040.26      7250784.21        2202829.        7250260.
      2202025.28       7249765.1
#Sta/Elev= 30
  3691.9  991.83  3743.4  988.91  3869.6   980.6  4167.8  967.26  4267.2  964.63
  4319.6   965.5  4357.9  961.76  4532.3  957.09  4705.6  956.81  4837.9  956.27
  4903.3  957.11  4926.8  959.42  4957.2  958.28  4968.1  956.71  4979.2  950.85
  4990.2  949.09  4992.7  948.59  5015.2  949.09  5019.4  954.31  5026.8  957.81
  5317.1  956.08  5446.5  958.11  5483.2  955.28  5498.6  959.45    5575  957.96
  5629.9  956.96    5705  962.79  5840.5  973.31  5855.9  976.56  5955.6  980.53
#Mann= 9 ,-1 , 0
  3691.9     .16       0  3743.4     .05       0  4705.6     .05       0
  4837.9     .05       0  4990.2    .035       0  5015.2     .05       0
  5026.8     .05       0    5575     .05       0    5705     .16       0
Bank Sta=4990.2,5015.2
XS Rating Curve= 0 ,0
Exp/Cntr=0.3,0.1

Type RM Length L Ch R = 1 ,516694  ,504,504,504
BEGIN DESCRIPTION:
Denton Creek 254.0
END DESCRIPTION:
XS GIS Cut Line= 3
      2203828.99        7250010.        2203029.        7249810.
      2202278.97      7249259.98
#Sta/Elev= 30
  4195.8  993.41  4471.5  976.04  4593.4  968.66  4649.3   965.2  4708.6  964.26
  4713.8   962.4    4755  961.12  4796.2   956.7  4886.9  955.17  4968.9  957.33
    4985  951.52  4989.5  950.72  4989.9  948.14  4992.4  947.64  5014.9  948.14
  5017.8  955.22  5049.6  956.39  5178.2  955.11  5192.9  952.02  5199.1  957.13
    5220  959.82  5234.6  956.62    5258  955.16  5479.2  954.74  5656.8  957.33
  5757.1  963.43  5771.8  968.15  5809.1   968.1  5818.5  969.76  5950.5  981.89
#Mann= 11 ,-1 , 0
  4195.8     .16       0  4471.5     .05       0  4593.4     .05       0
  4886.9     .05       0    4985     .05       0  4989.9    .045       0
  5014.9     .05       0  5049.6     .05       0    5258     .05       0
  5809.1     .05       0  5818.5     .05       0
Bank Sta=4989.9,5014.9
XS Rating Curve= 0 ,0
Exp/Cntr=0.3,0.1

Type RM Length L Ch R = 1 ,516190  ,482,482,482
BEGIN DESCRIPTION:
Denton Creek 253.0
END DESCRIPTION:
XS GIS Cut Line= 3
      2203829.01      7249910.01        2203279.        7249410.
      2201679.04      7248710.02
#Sta/Elev= 30
  4229.6  990.32    4534  969.46  4625.9   968.4  4658.3  963.23  4760.4  954.61
  4904.5  954.96  4965.8  955.24  4981.9  952.44  4992.8  946.96  4995.3  946.46
  5017.8  946.96  5039.6  957.31  5081.5   953.9  5639.1  954.76  5726.1   957.6
  5737.4  961.91  5747.9  966.04  5769.7   962.4  5796.5  967.17  5878.5  972.49
  6011.8  972.41  6195.7  983.41  6308.9  988.46  6315.5  991.53  6337.7  989.97
  6384.5  996.26  6460.1  996.96  6559.1 1001.57  6605.9  1007.1  6719.3 1011.36
#Mann= 9 ,-1 , 0
  4229.6     .16       0  4658.3     .05       0  4904.5     .05       0
  4992.8    .035       0  5017.8     .05       0  5081.5     .05       0
  5737.4     .05       0  5796.5     .05       0  6195.7     .05       0
Bank Sta=4992.8,5017.8
XS Rating Curve= 0 ,0
Exp/Cntr=0.3,0.1

Type RM Length L Ch R = 1 ,515708  ,575,575,575
BEGIN DESCRIPTION:
Denton Creek 252.0
END DESCRIPTION:
XS GIS Cut Line= 3
      2203929.04      7249260.02        2203529.        7249010.
      2201929.03      7248460.01
#Sta/Elev= 30
    4503  980.05  4593.7  969.54  4786.1  957.86  4961.2  954.58  4977.4  953.12
  4983.4  945.92  4985.9  945.42  5008.4  945.92  5016.3  950.82  5038.2  957.82
  5047.6  955.81  5059.3  957.58  5091.1  952.81  5640.4  954.06  5746.7   955.8
  5778.4  960.74  5792.1  957.24  5799.5  959.79  5911.8  960.92  5958.2  966.22
  6062.7  970.41    6085  968.22  6099.2  974.32  6125.2  973.46  6130.5  975.39
  6148.5  973.46  6275.4  983.23  6286.7  981.88  6343.9  987.06  6666.6 1003.47
#Mann= 5 ,-1 , 0
    4503     .16       0  4593.7     .05       0  4983.4    .045       0
  5008.4     .05       0  5640.4     .05       0
Bank Sta=4983.4,5008.4
XS Rating Curve= 0 ,0
Exp/Cntr=0.3,0.1

Type RM Length L Ch R = 1 ,515133  ,535,535,535
BEGIN DESCRIPTION:
Denton Creek 251.0
END DESCRIPTION:
XS GIS Cut Line= 3
      2203979.03      7248660.02        2203629.        7248460.
      2202479.01        7248210.
#Sta/Elev= 30
  4630.5  980.04  4665.8  971.19  4689.1  967.64  4768.7  959.26  4890.7  953.14
  4963.3  954.54  4976.1  954.25  4988.3  949.09  4991.6  945.84  4994.1  945.34
  5016.6  945.84    5020  952.02  5053.1  954.88  5064.4  952.88  5102.2  952.01
    5136  953.31  5330.4  951.74  5371.4  952.67  5607.8  951.73  5671.2  951.45
  5688.6  953.44  5698.8   956.7  5709.1  957.26  5759.2  955.71  5780.7   958.6
  5862.6  964.72  5999.7  971.46  6087.7  977.58  6118.4  981.49  6210.5  985.69
#Mann= 7 ,-1 , 0
  4630.5     .05       0  4689.1     .05       0  4890.7     .05       0
  4963.3     .05       0  4991.6    .045       0  5016.6     .05       0
  5607.8     .05       0
Bank Sta=4991.6,5016.6
XS Rating Curve= 0 ,0
Exp/Cntr=0.3,0.1

Type RM Length L Ch R = 1 ,514598  ,594,594,594
BEGIN DESCRIPTION:
Denton Creek 250.0
END DESCRIPTION:
XS GIS Cut Line= 3
      2204220.15      7248014.95        2203679.        7247960.
      2202152.34      7247515.47
#Sta/Elev= 30
  4441.9  978.87  4563.7  975.59  4740.9  964.69  4794.9  957.96  4930.4  953.71
  4945.6  955.48  4975.8  950.78  4983.3     947  4983.8   944.2  4986.3   943.7
  5008.8   944.2  5017.1   952.2  5027.5   952.6  5470.4  950.92  5558.7  950.35
  5652.6  953.45  5714.4  959.01  5777.4  959.61  5871.1  968.83  5964.6  973.95
  6071.4  968.65  6141.9  965.48  6181.2  961.32  6258.7  967.21  6291.3  965.99
  6330.9   967.3  6359.2  971.98  6364.4  969.67  6397.9  976.51  6575.9  989.53
#Mann= 8 ,-1 , 0
  4441.9     .16       0  4740.9     .05       0  4930.4     .05       0
  4983.8    .045       0  5008.8     .05       0  5470.4     .05       0
  6071.4     .16       0  6291.3     .05       0
Bank Sta=4983.8,5008.8
XS Rating Curve= 0 ,0
Exp/Cntr=0.3,0.1

Type RM Length L Ch R = 1 ,514004  ,129,129,129
BEGIN DESCRIPTION:
Denton Creek299
END DESCRIPTION:
XS GIS Cut Line= 3
      2204178.61      7247754.93       2203602.6      7247213.87
      2202257.38      7246779.78
#Sta/Elev= 30
  4455.8  973.47  4747.5  959.02  4933.1  949.97  4975.6  951.56  4977.3  943.39
  4979.8  942.89  5002.3  943.39    5025   949.4  5053.3   952.1  5138.3  948.55
    5243  950.73  5291.9  950.81  5344.9  947.16  5371.7  950.04  5467.8  952.57
  5757.6   956.2  5979.4  959.41  6476.9  978.91  6489.8  978.93  6500.3  974.39
  6521.3  971.08    6573  977.37  6578.3  981.45  6584.3   982.5  6605.1  982.69
  6610.3  977.95  6615.9  977.21  6626.4  978.63  6642.4     985  6659.6  978.49
#Mann= 7 ,-1 , 0
  4455.8     .05       0  4747.5     .16       0  4977.3     .07       0
  5002.3     .16       0    5243     .05       0  5757.6     .16       0
  5979.4     .05       0
Bank Sta=4977.3,5002.3
XS Rating Curve= 0 ,0
Exp/Cntr=0.3,0.1

Type RM Length L Ch R = 1 ,513875  ,666,666,666
BEGIN DESCRIPTION:
Denton Creek298
END DESCRIPTION:
XS GIS Cut Line= 3
      2204230.06      7247651.36      2203690.16      7247136.59
       2202273.4      7246658.89
#Sta/Elev= 30
  4432.9  974.57  4449.5   974.2  4619.1  964.82  4802.5  954.37    4944  953.27
  4972.3  950.92  4979.2  948.76  4980.9  942.61  4983.4  942.11  5005.9  942.61
  5014.7  949.24  5042.7  953.89  5141.8  949.83  5164.2  953.64  5310.5  947.12
  5820.4  955.64  5929.3  960.74  6003.2  964.83  6055.5  961.13  6108.8  966.53
  6129.9   962.3  6275.8  970.28  6433.2  972.86    6457  968.31  6488.7  974.68
  6541.5  975.93  6564.4   971.9  6604.8  978.79  6627.4  972.69    6674   982.2
#Mann= 8 ,-1 , 0
  4432.9     .16       0  4449.5     .05       0  4619.1     .16       0
  4980.9     .07       0  5005.9     .16       0  5164.2     .05       0
  5820.4     .16       0  5929.3     .05       0
Bank Sta=4980.9,5005.9
XS Rating Curve= 0 ,0
Exp/Cntr=0.3,0.1

Type RM Length L Ch R = 1 ,513209  ,920,920,920
BEGIN DESCRIPTION:
Denton Creek 247.0
END DESCRIPTION:
XS GIS Cut Line= 3
      2204921.18      7247327.47      2204078.19      7246619.95
      2201969.23      7245530.91
#Sta/Elev= 30
  4091.4  980.91  4217.9  975.69  4247.6  978.11    4297  975.54  4303.6  972.14
  4381.6   972.5  4493.7  962.68  4926.4  949.52  4985.2  946.51    4987  941.68
  4989.5  941.18    5012  941.68  5013.8   947.7  5021.2  949.99    5125  949.91
  5720.6  946.95  5898.3  947.56  6046.4  949.82  6401.2  974.75  6528.5   973.3
  6683.5  961.59    6823  961.42  7082.3  967.52  7314.7  978.91  7386.8  977.44
  7403.3  981.91  7408.9  978.57  7453.2  978.92  7498.2  988.16  7565.5  990.05
#Mann= 9 ,-1 , 0
  4091.4     .05       0  4217.9     .16       0  4493.7     .05       0
  4926.4     .16       0    4987     .07       0    5012     .16       0
    5125     .05       0  5720.6     .16       0  5898.3     .05       0
Bank Sta=4987,5012
XS Rating Curve= 0 ,0
Exp/Cntr=0.3,0.1

Type RM Length L Ch R = 1 ,512289  ,963,963,963
BEGIN DESCRIPTION:
Denton Creek 245.0
END DESCRIPTION:
XS GIS Cut Line= 3
      2205329.04      7246310.02       2204056.2       7245667.4
      2202183.32      7245091.09
#Sta/Elev= 30
  4249.1   973.4  4370.5   966.4  4473.9  962.34  4764.4  947.99  4865.1  946.92
    4971  948.95  4977.3  948.15  4987.2  939.55  4989.7  939.05  5012.2  939.55
  5022.1  947.01  5032.3  947.69  5126.4  946.72  5143.7     948  5232.9   944.6
  5313.4  944.13  5490.8   946.1  6635.2  950.27  7092.9  956.27  7293.8  961.96
    7345  967.62  7350.2  966.05    7367  968.09  7415.6  967.46  7448.3  970.08
  7471.6  965.44  7501.8  966.86  7512.3  969.03    7519  972.09  7634.5  977.69
#Mann= 12 ,-1 , 0
  4249.1     .16       0  4370.5     .05       0  4473.9     .16       0
  4865.1     .05       0  4987.2    .035       0  5012.2     .05       0
  5126.4     .16       0  5490.8     .05       0  6635.2     .05       0
  7092.9     .05       0  7501.8     .16       0  7512.3     .05       0
Bank Sta=4987.2,5012.2
XS Rating Curve= 0 ,0
Exp/Cntr=0.3,0.1

Type RM Length L Ch R = 1 ,511326  ,539,539,539
BEGIN DESCRIPTION:
Denton Creek 244.0
END DESCRIPTION:
XS GIS Cut Line= 3
      2205378.99      7245959.99        2204729.        7245160.
      2203929.02      7244360.02
#Sta/Elev= 30
  3958.8  971.13  4108.2  963.46    4369  946.92  4421.4  944.18  4563.6  943.62
  4641.7  945.86  4654.8  944.78  4726.7  945.78    4797  944.73  4953.6  946.99
  4989.6  940.71  4990.8  938.14  4993.4  937.64  5016.6  938.14  5017.8  944.81
    5032  946.85  5097.8  945.34    5131  946.72  5159.3  944.02  5314.8  942.95
  5369.7  944.12  5470.4  943.08  5605.8  945.99  5653.4  947.31  5742.5  949.88
  5795.2  953.49  5879.1  960.22  5937.1  964.47  6078.5  976.84  6120.9  979.04
#Mann= 12 ,-1 , 0
  3958.8     .16       0    4369     .05       0  4990.8    .035       0
  5016.6     .05       0  5097.8     .05       0  5369.7     .05       0
  5605.8     .05       0  5653.4     .05       0  5742.5     .05       0
  5795.2     .05       0  5879.1     .05       0  5937.1     .05       0
Bank Sta=4990.8,5016.6
XS Rating Curve= 0 ,0
Exp/Cntr=0.3,0.1

Type RM Length L Ch R = 1 ,510787  ,812,812,812
BEGIN DESCRIPTION:
Denton Creek 243.0
END DESCRIPTION:
XS GIS Cut Line= 3
      2205479.01      7246060.05        2205129.        7244810.
      2204579.03      7244010.04
#Sta/Elev= 30
  3722.7  979.18  3782.6  976.04  3965.3  965.79  4273.1  944.35  4321.4   943.4
    4512  942.77  4563.9  946.07  4584.7  944.03  4665.5  943.35  4918.2  945.25
  4964.4   946.3  4979.3  941.24  4985.7  935.06  4988.3  934.56  5011.5  935.06
  5018.2  941.95  5020.5  941.95  5023.9  941.95  5028.3  945.67  5043.2  945.97
  5222.4  942.15  5258.3  944.86  5279.2  942.23  5503.2  946.43  5566.9  951.74
  5616.8  950.47  5639.7  957.01  5688.5  962.19  5825.9  961.22  5991.6  967.41
#Mann= 7 ,-1 , 0
  3722.7     .05       0  3782.6     .16       0  4321.4     .05       0
  4918.2     .16       0  4985.7     .07       0  5011.5     .16       0
  5020.5     .05       0
Bank Sta=4985.7,5011.5
XS Rating Curve= 0 ,0
Exp/Cntr=0.3,0.1

Type RM Length L Ch R = 1 ,509975  ,852,852,852
BEGIN DESCRIPTION:
Denton Creek 242.0
END DESCRIPTION:
XS GIS Cut Line= 3
       2206266.1      7245848.26      2206185.98      7244921.23
      2204964.74      7243554.17
#Sta/Elev= 30
    3348  972.87  3366.3  975.41  3396.4  970.12  3456.7  963.89  3490.1  964.08
  3516.9  959.41  3697.6   949.8  3980.9  945.53  4139.7  944.85  4227.4  943.66
  4461.4  941.54  4561.3  943.59  4716.3  941.25  4936.2  944.49  4957.1  939.94
  4985.5  937.96  4993.5  934.25  4996.1  933.75  5019.4  934.25  5020.7  937.69
  5028.2  941.17  5042.4  943.92  5183.7  942.46  5247.2  939.13  5283.1  942.61
  5502.2  946.25  5587.4  951.97  5658.5  953.15  5807.3  966.26  6111.6  984.73
#Mann= 7 ,-1 , 0
    3348     .05       0  3980.9     .16       0  4139.7     .05       0
  4227.4     .16       0  4561.3     .05       0  4993.5    .035       0
  5019.4     .05       0
Bank Sta=4993.5,5019.4
XS Rating Curve= 0 ,0
Exp/Cntr=0.3,0.1

Type RM Length L Ch R = 1 ,509123  ,1190,1190,1190
BEGIN DESCRIPTION:
Denton Creek297
END DESCRIPTION:
XS GIS Cut Line= 3
      2207265.31      7245050.51      2206598.02      7244110.44
       2205460.9      7242967.76
#Sta/Elev= 30
    3412   964.7  3487.9  959.58  3523.5   959.6  3532.2  957.64  3607.8  954.65
    3761  945.18  3815.2  943.63  3983.6   944.2  4120.2  942.56  4191.5  944.42
  4320.1  941.79  4565.6   941.1    4700  939.83  4727.1  941.38  4748.3  939.19
  4771.5  939.46  4967.5  941.47  4974.6  937.01  4975.7  932.68  4978.3  932.18
  5001.6  932.68    5017  934.83  5052.4   934.9  5101.8  942.04  5405.9  937.52
  5731.2  943.17  5738.2  944.83  5759.5  944.24  5929.2  953.81  6176.9  974.34
#Mann= 8 ,-1 , 0
    3412     .16       0  3607.8     .05       0  3815.2     .16       0
  4565.6     .05       0    4700     .16       0  4771.5     .05       0
  4975.7     .05       0  5001.6     .05       0
Bank Sta=4975.7,5001.6
XS Rating Curve= 0 ,0
Exp/Cntr=0.3,0.1

Type RM Length L Ch R = 1 ,507933  ,993,993,993
BEGIN DESCRIPTION:
Denton Creek 241.0
END DESCRIPTION:
XS GIS Cut Line= 3
      2207421.08      7244575.45      2206952.91      7243186.66
        2206429.        7242010.
#Sta/Elev= 30
  3321.5  971.92  3499.3  967.86  3563.7  967.61  3879.3  945.38    3973  938.27
  4044.8  938.16  4093.7  946.24  4108.2  944.96  4125.1  939.22  4150.4  937.98
  4496.5  936.21    4583  935.96  4604.2  933.84  4635.8  937.06  4713.7  936.22
  4833.1   935.6  4969.5  939.87  4983.5  936.88  4987.7  929.22  4990.4  928.72
  5014.8  929.22  5035.5  939.66  5341.7  937.37  5363.6  934.22  5377.2  938.05
    5484   936.7  5620.5  939.42  5788.7  947.22  5840.7  954.39  6075.1  977.11
#Mann= 8 ,-1 , 0
  3321.5     .16       0  3499.3     .05       0  3879.3     .05       0
  4496.5     .16       0  4713.7     .05       0  4987.7     .05       0
  5014.8     .05       0  5620.5     .05       0
Bank Sta=4987.7,5014.8
XS Rating Curve= 0 ,0
Exp/Cntr=0.3,0.1

Type RM Length L Ch R = 1 ,506940  ,1473,1473,1473
BEGIN DESCRIPTION:
Denton Creek 239.0
END DESCRIPTION:
XS GIS Cut Line= 4
      2207895.94      7244094.12      2207845.71       7243054.8
      2207557.12      7241892.46      2207167.93      7241577.87
#Sta/Elev= 30
  3431.8  958.31  3476.5  957.64  3776.3  934.93  3968.1  934.53  4086.7  931.51
  4166.8  933.34  4186.8  931.04    4327  934.68  4487.6  941.72    4570  935.25
  4714.3   932.6  4971.9  938.45  4982.4  938.15    4994  929.67  4999.5  928.37
  5002.2  927.87  5026.6  928.37  5033.7  936.62    5044  937.82  5106.4  935.74
    5404   935.9  5538.6  935.46  5641.5  939.75  5762.7  947.21  5797.9  952.57
  5884.2  961.35  5948.1  964.71  6018.5  971.48  6126.7  975.38  6170.4  975.06
#Mann= 8 ,-1 , 0
  3431.8     .05       0  3968.1     .05       0    4994     .05       0
  4999.5    .035       0  5026.6     .05       0    5404     .16       0
  5641.5     .05       0  6126.7     .05       0
Bank Sta=4999.5,5026.6
XS Rating Curve= 0 ,0
Exp/Cntr=0.3,0.1

Type RM Length L Ch R = 1 ,505467  ,1103,1103,1103
BEGIN DESCRIPTION:
Denton Creek 237.0
END DESCRIPTION:
XS GIS Cut Line= 3
      2208920.16      7244803.14        2209079.        7242710.
      2209051.29       7241825.7
#Sta/Elev= 30
  2895.7   971.7  3081.5  967.44  3706.3   941.1    3747  939.41  3889.6  933.38
  3941.8  931.16  4179.1  930.76  4292.9  932.04    4333  928.84    4353  930.61
  4373.1  929.04  4413.2  931.74  4460.9  930.88  4535.4  932.48  4669.4  931.97
  4945.4  934.69  4964.8  935.06  4990.6  926.21  4993.4  925.71  5019.2  926.21
  5024.9   935.4  5030.3  935.68  5094.9  933.12  5152.2  935.64    5285  933.21
    5325  936.74  5405.1  940.11  5425.1  943.75  5543.4  952.45  5879.6  972.97
#Mann= 12 ,-1 , 0
  2895.7     .05       0  3706.3     .05       0    3747     .05       0
  3889.6     .05       0  4179.1     .12       0  4460.9     .05       0
  4669.4     .05       0  4945.4     .16       0  4990.6     .07       0
  5019.2     .16       0  5030.3     .05       0  5543.4     .16       0
Bank Sta=4990.6,5019.2
XS Rating Curve= 0 ,0
Exp/Cntr=0.3,0.1

Type RM Length L Ch R = 1 ,504364  ,1069,1069,1069
BEGIN DESCRIPTION:
Denton Creek 235.0
END DESCRIPTION:
XS GIS Cut Line= 3
      2209558.47       7245725.7        2210129.        7242860.
      2210128.73      7241254.34
#Sta/Elev= 30
  2072.2  978.49  2465.5  955.07  2965.3  951.42  3013.5  951.83    3118  951.46
  3199.6  940.36  3292.4  937.28  3383.2  936.18  3482.4  935.61  3581.6  935.33
  3605.7  934.77  3674.8   931.7    3702  931.44    3922  928.66  4147.8  929.65
  4270.4  928.92  4771.8  930.78  4772.1  930.78  4870.9  931.78  4973.8  933.07
  4989.8  924.18  4992.6  923.68  5018.4  924.18  5024.1  930.82  5044.1  933.52
  5364.1  928.35  5792.9  934.91  6002.2  943.47  6394.1  975.88  6599.8  977.85
#Mann= 20 ,-1 , 0
  2072.2     .05       0  2965.3     .05       0  3013.5     .05       0
  3292.4     .05       0  3383.2     .05       0  3482.4     .12       0
  3581.6     .05       0  3605.7     .12       0  3674.8     .05       0
    3702     .12       0    3922     .05       0  4147.8     .16       0
  4270.4     .05       0  4771.8     .05       0  4772.1     .05       0
  4870.9     .05       0  4989.8     .05       0  5018.4     .05       0
  5792.9     .05       0  6002.2     .16       0
Bank Sta=4989.8,5018.4
XS Rating Curve= 0 ,0
Exp/Cntr=0.3,0.1

Type RM Length L Ch R = 1 ,503295  ,1051,1051,1051
BEGIN DESCRIPTION:
Denton Creek 233.0
END DESCRIPTION:
XS GIS Cut Line= 3
      2210696.98      7245691.02      2211197.84      7242742.37
        2211179.      7241710.03
#Sta/Elev= 30
  2460.4  969.91  2620.2  962.63  2877.4  944.27    3137  930.81  3587.3  925.05
  3597.5  929.87  3607.6  930.61  3668.5  925.01  3701.4  925.24  3760.6  924.89
  3769.9  928.71  3995.4  927.03  4379.8  928.22  4413.6  929.25  4429.2  925.46
  4594.1  926.91  4918.9   930.1  4966.8  931.82    4977  929.87  4982.9  921.01
  4985.7  920.51  5011.5  921.01  5017.5  928.86  5045.8  931.05  5307.8  928.11
  5503.7  940.53  5743.7  947.53  6013.7  948.25  6263.8  961.23  6483.8  967.48
#Mann= 11 ,-1 , 0
  2460.4     .05       0  2877.4     .05       0    3137     .16       0
  3701.4     .05       0  3995.4     .05       0  4379.8     .16       0
  4594.1     .05       0  4918.9     .05       0  4982.9    .035       0
  5011.5     .05       0  5045.8     .16       0
#XS Ineff= 2 , 0
       0  3949.8  952.05               0
Permanent Ineff=
       F       F
Bank Sta=4982.9,5011.5
XS Rating Curve= 0 ,0
Exp/Cntr=0.3,0.1

Type RM Length L Ch R = 1 ,502244  ,639,639,639
BEGIN DESCRIPTION:
Denton Creek 231.0
END DESCRIPTION:
XS GIS Cut Line= 3
       2211872.4      7245570.01      2211868.76      7244141.42
        2211679.      7241909.97
#Sta/Elev= 30
  2101.2  957.16  2111.2  957.09  2120.1  954.67  2151.2  943.21  2161.2  941.94
  2311.2  937.08  2811.2  937.51  3431.2  932.41  3772.1  927.07  4083.2  927.12
  4113.3  923.51  4123.4  926.52  4178.4  926.75  4253.8  928.77  4424.4  926.62
  4665.3  926.79  4956.3  929.86  4976.4  927.76  4986.5  922.06  4987.5  919.76
  4990.3  919.26  5016.1  919.76  5016.6  925.99  5026.6   929.7  5177.1  928.19
  5327.7   934.6  5387.9  939.86  5592.9  951.54    5699  961.15  5769.3  965.11
#Mann= 5 ,-1 , 0
  2101.2     .05       0  2120.1     .05       0  4178.4     .16       0
  4987.5     .07       0  5016.1     .16       0
Bank Sta=4987.5,5016.1
XS Rating Curve= 0 ,0
Exp/Cntr=0.3,0.1

Type RM Length L Ch R = 1 ,501605  ,144,144,144
BEGIN DESCRIPTION:
Denton Creek296
END DESCRIPTION:
XS GIS Cut Line= 5
      2213331.71       7244351.7      2212801.37      7243542.46
      2212529.17      7243107.47      2212224.14      7242222.03
      2212048.28      7241510.73
#Sta/Elev= 30
  2912.1  945.13  3450.7  928.31  4063.7  925.27    4326  922.12  4354.4  924.85
  4495.7  921.37    4683  927.08  4728.6  925.42  4750.7  927.86  4951.2  928.64
  4963.9  928.82  4989.2  919.46    4992  918.96    5018  919.46  5021.1  927.57
  5052.3  927.09  5057.6  923.71  5098.7  928.54  5113.4   927.4  5172.5  928.75
  5246.8  933.85  5444.7  934.43  5506.5  940.75  5691.9   945.6    5764  952.43
  5805.2  950.36  5897.9  957.31  5939.1  955.87  5996.2  962.14    6062   964.9
#Mann= 7 ,-1 , 0
  2912.1     .05       0  4063.7     .05       0  4951.2     .05       0
  4989.2    .035       0    5018     .05       0  5113.4     .16       0
  5172.5     .05       0
#XS Ineff= 2 , 0
       0  3936.5   940.2               0
Permanent Ineff=
       F       F
Bank Sta=4989.2,5018
XS Rating Curve= 0 ,0
Exp/Cntr=0.3,0.1

Type RM Length L Ch R = 1 ,501461  ,431,431,431
BEGIN DESCRIPTION:
Denton Creek295
END DESCRIPTION:
XS GIS Cut Line= 5
      2213507.19      7244162.61      2212984.34      7243318.74
      2212624.41      7242978.33      2212369.34      7242197.16
      2212171.81      7241477.04
#Sta/Elev= 30
  3003.4  953.39  3562.7  935.88  3809.6  934.31  3977.4  941.48  4119.2  940.94
  4161.7  940.08  4289.1  931.68  4338.5  932.11  4354.8  927.95  4388.2  921.62
  4458.6  923.71  4573.9  922.34  4742.2  927.63  4836.9   926.3  4916.2  927.75
  4977.5  927.55  4984.2  919.55  4989.7  917.32  4992.6  916.82  5018.5  917.32
  5026.3  925.97    5036  929.42  5110.4   928.9    5137  926.48  5448.6  934.23
  5596.8  941.12  5670.9  942.35  5750.2  950.57  5824.3  954.48    6060  963.18
#Mann= 5 ,-1 , 0
  3003.4     .05       0  4354.8     .05       0  4916.2     .05       0
  4989.7    .035       0  5018.5     .05       0
Bank Sta=4989.7,5018.5
XS Rating Curve= 0 ,0
Exp/Cntr=0.3,0.1

Type RM Length L Ch R = 1 ,501030  ,923,923,923
BEGIN DESCRIPTION:
Denton Creek 229.0
END DESCRIPTION:
XS GIS Cut Line= 4
      2213651.65      7244232.97      2213166.06      7243259.52
      2212747.48      7242052.85      2212397.21       7241523.5
#Sta/Elev= 30
  3010.9  951.41  3208.5  952.17  3617.7  935.55  3784.7  932.77  3986.1  935.96
  4166.5  946.71  4259.9  947.49  4353.3  942.56  4467.3   931.5  4534.9  927.97
  4560.7  919.21  4616.9  919.16  4626.9  921.69  4695.6  923.28  4835.7  923.74
  4940.5  926.18  4976.8  927.76  4983.5  916.86  4986.4  916.36  5012.3  916.86
  5029.7  926.62  5241.4  924.19  5273.1  927.99  5297.3  926.55  5471.1  934.47
  5621.5  945.95  5630.6  948.67    5760  955.77  5853.2  959.55  6010.7  960.87
#Mann= 7 ,-1 , 0
  3010.9     .05       0  4626.9     .12       0  4695.6     .05       0
  4835.7     .16       0  4940.5     .05       0  4983.5    .035       0
  5012.3     .05       0
Bank Sta=4983.5,5012.3
XS Rating Curve= 0 ,0
Exp/Cntr=0.3,0.1

Type RM Length L Ch R = 1 ,500107  ,1393,1393,1393
BEGIN DESCRIPTION:
Denton Creek 227.0
END DESCRIPTION:
XS GIS Cut Line= 3
      2214978.98      7243259.98        2213429.        7241860.
      2212728.98      7241209.99
#Sta/Elev= 30
  2956.5  963.08  3423.9  935.09  3586.8   929.4  3603.3  926.64  3846.4   919.5
  4216.8  919.85  4251.9  922.57  4287.8  921.89  4464.9  922.04  4535.1  920.07
  4749.5  922.62  4885.4  924.59    4967  924.56  4974.5  917.54    4988   914.6
  4990.9   914.1  5017.8   914.6  5023.8  915.03  5031.3  919.63    5038  918.49
  5041.8  922.29  5052.2   924.3    5177  921.28  5208.1  921.28  5335.1  928.97
  5420.1  937.97  5561.9  939.76  5717.2  947.15  5908.3  952.69  6000.4  958.44
#Mann= 9 ,-1 , 0
  2956.5     .05       0  3603.3     .05       0  3846.4     .16       0
  4287.8     .05       0  4749.5     .05       0  4885.4     .16       0
    4988     .07       0  5017.8     .16       0    5177     .05       0
Bank Sta=4988,5017.8
XS Rating Curve= 0 ,0
Exp/Cntr=0.3,0.1
