HEC-RAS study Denton Creek.prj: Denton Creek Base Level Engineering

--- Denton Creek.g01 (geometry) --- (continued)

Type RM Length L Ch R = 1 ,498714  ,134,134,134
BEGIN DESCRIPTION:
Denton Creek294
END DESCRIPTION:
XS GIS Cut Line= 6
      2215313.35      7241363.98      2214651.11      7241049.36
       2214286.1      7240975.12      2214031.35      7241258.89
      2213731.66      7241335.95      2212557.34      7240343.93
#Sta/Elev= 30
  3949.4  957.66  4339.7  935.96  4362.4  940.63  4385.1  935.43  4464.4   935.1
    4746  920.18  4803.4  923.61  4899.3  916.12    4950  916.31  4960.3  919.75
  4970.5  917.59  4975.9  912.48  4978.9  911.98  5005.8  912.48    5027  922.02
  5346.6  924.87  5360.8  921.94  5707.5  922.43  5753.7  928.75  5760.3  925.07
  5791.1  927.46  5797.6   926.1  5911.3  922.32  6283.1  921.05    6410  925.68
  6424.2  921.75  6474.4  921.48  6558.9  926.17  7090.7  933.21  7294.1  945.19
#Mann= 9 ,-1 , 0
  3949.4     .05       0  4899.3     .16       0  4975.9     .07       0
  5005.8     .16       0    5027     .05       0  5791.1     .16       0
  5797.6     .05       0  5911.3     .16       0  6283.1     .05       0
Bank Sta=4975.9,5005.8
XS Rating Curve= 0 ,0
Exp/Cntr=0.3,0.1

Type RM Length L Ch R = 1 ,498580  ,1076,1076,1076
BEGIN DESCRIPTION:
Denton Creek293
END DESCRIPTION:
XS GIS Cut Line= 6
      2215341.07      7241221.35      2214552.81      7240866.06
      2214207.26      7240855.47      2213932.08      7241202.57
      2213745.62      7241248.76      2212597.06      7240200.27
#Sta/Elev= 30
  3961.6  955.26  4128.5  943.28  4192.4  942.33  4295.9  936.74  4440.2  934.72
  4561.4  936.31  4720.7  922.52  4809.2  920.02  4930.1  920.58  4940.1  919.23
  4945.1  911.59  4948.1  911.09  4975.1  911.59  5000.1  911.81  5020.1  921.53
  5090.2  920.01  5110.2  922.63  5120.2   920.2  5195.1  919.23  6140.1  919.32
  6140.2  919.32  6369.4  919.43  6702.6  927.66  6979.5  929.44  7000.3  927.36
  7028.9  931.57  7085.7  931.26  7194.1  941.47  7350.1  952.96  7363.4  953.86
#Mann= 7 ,-1 , 0
  3961.6     .05       0  4945.1    .035       0  4975.1     .05       0
  6140.1     .16       0  6140.2     .05       0  7194.1     .16       0
  7350.1     .05       0
Bank Sta=4945.1,4975.1
XS Rating Curve= 0 ,0
Exp/Cntr=0.3,0.1

Type RM Length L Ch R = 1 ,497504  ,1028,1028,1028
BEGIN DESCRIPTION:
Denton Creek 223.0
END DESCRIPTION:
XS GIS Cut Line= 3
      2215727.56      7241089.38        2214929.        7240010.
      2213234.93      7238498.83
#Sta/Elev= 30
  3659.8  954.18  3830.4  948.53  3873.6  943.02  3936.9  942.44  4007.7  935.61
  4151.9  925.97  4469.2  916.83  4815.9  918.23  4844.9  921.33    4903  919.98
  4943.2  913.02  4959.7  914.43  4979.7  908.08  4982.7  907.58  5010.7  908.08
    5038  920.54  5349.8  915.46  5427.6  917.98  5823.9  914.24  6156.6  915.37
    6267   921.4  6447.6   926.3  6482.7  924.05  6511.1  927.73  6829.7  921.55
  7146.8  924.76  7184.1  924.82  7219.3  934.11  7240.3  935.43  7272.6  947.29
#Mann= 9 ,-1 , 0
  3659.8     .05       0  3873.6     .16       0  4007.7     .05       0
  4469.2     .16       0  4943.2     .05       0  4979.7    .035       0
  5010.7     .05       0    6267     .16       0  7146.8     .05       0
Bank Sta=4979.7,5010.7
XS Rating Curve= 0 ,0
Exp/Cntr=0.3,0.1

Type RM Length L Ch R = 1 ,496476  ,1186,1186,1186
BEGIN DESCRIPTION:
Denton Creek 221.0
END DESCRIPTION:
XS GIS Cut Line= 3
      2216016.56      7240678.89      2215981.47      7240059.61
      2214710.65      7237629.17
#Sta/Elev= 30
  3598.1  944.46    3733  941.26  3895.8  931.48  4187.9  918.92  4317.3  917.97
  4433.4   913.7  4538.1  912.57    4709   916.8  4798.1     916  4835.9  914.34
  4857.9  916.44  4968.3  916.34  4984.7  911.41  4991.3  904.69  4994.3  904.19
  5022.3  904.69  5024.9   909.3  5028.9  916.39    5073  914.48  5287.5  915.74
  5332.3  916.81  5337.9  914.74  5436.7  915.08  5470.5  913.01    6298  914.76
  6347.3  917.89  6479.7     919  6506.1   921.7  6827.3  945.15    6961  958.55
#Mann= 10 ,-1 , 0
  3598.1     .05       0    3733     .16       0  3895.8     .05       0
  4798.1     .16       0  4991.3     .07       0  5022.3     .16       0
  5024.9     .05       0  5287.5     .05       0    6298     .05       0
  6506.1     .16       0
#XS Ineff= 2 , 0
       0                  5898.7       0  938.66
Permanent Ineff=
       F       F
Bank Sta=4991.3,5022.3
XS Rating Curve= 0 ,0
Exp/Cntr=0.3,0.1

Type RM Length L Ch R = 1 ,495290  ,1070,1070,1070
BEGIN DESCRIPTION:
Denton Creek 219.0
END DESCRIPTION:
XS GIS Cut Line= 3
      2216667.97      7240675.99        2216529.        7238760.
      2216263.56      7238096.01
#Sta/Elev= 30
  3056.2  941.71  3202.6  935.94  3332.9  925.78  3382.8  924.47  3393.1  922.23
  3467.1  918.02  3573.5  910.82  3964.6  910.54  4165.1  913.08  4245.3  912.23
  4295.4  914.41  4536.3  913.97    4699  913.43    4897  912.41  4910.1  909.84
  4922.1  911.99  4947.1  912.54  4967.2  907.54  4971.1  901.35  4974.1  900.85
  5002.1  901.35  5009.5  902.01  5021.7  913.17  5040.5  912.55  5063.4  915.14
  5315.2  924.12  5584.5  931.84  5623.4  930.96  5638.4  933.43  5692.3  934.99
#Mann= 7 ,-1 , 0
  3056.2     .16       0  3467.1     .05       0  4536.3     .05       0
    4699     .16       0  4922.1     .05       0  4971.1    .035       0
  5002.1     .05       0
Bank Sta=4971.1,5002.1
XS Rating Curve= 0 ,0
Exp/Cntr=0.3,0.1

Type RM Length L Ch R = 1 ,494220  ,1076,1076,1076
BEGIN DESCRIPTION:
Denton Creek 217.0
END DESCRIPTION:
XS GIS Cut Line= 3
      2217370.71      7240911.62        2217529.        7238710.
        2217579.      7237559.99
#Sta/Elev= 30
  2785.6  941.67  2879.3   936.5  2885.4  936.17  2897.5  937.18  3117.4  924.56
  3147.2  921.96  3270.7  915.87  3448.9  908.79  3890.1  910.19  4040.4  907.76
  4063.8  911.14  4572.9  909.19  4812.4  909.58  4842.5  905.15  4872.6   909.9
  4920.4  908.45  4972.8  910.43  4982.9  905.82  4987.4  898.05  4990.4  897.55
  5018.4  898.05  5022.9  904.99  5042.9   909.5    5063  910.49  5233.1  911.22
  5253.1  902.15  5283.2  911.42  5352.2  910.43  5715.5  910.47    6144  932.53
#Mann= 12 ,-1 , 0
  2785.6     .05       0  2879.3     .16       0  2885.4     .05       0
  3117.4     .16       0  3147.2     .05       0  3270.7     .05       0
  4063.8     .05       0  4572.9     .16       0  4987.4     .07       0
  5018.4     .16       0  5352.2     .05       0  5715.5     .16       0
Bank Sta=4987.4,5018.4
XS Rating Curve= 0 ,0
Exp/Cntr=0.3,0.1

Type RM Length L Ch R = 1 ,493144  ,1035,1035,1035
BEGIN DESCRIPTION:
Denton Creek 216.0
END DESCRIPTION:
XS GIS Cut Line= 4
      2218302.34      7241625.27      2218664.54      7239540.65
        2218379.        7238560.      2217926.31       7236995.3
#Sta/Elev= 30
  1834.8  914.65    2547  912.84  2824.4  911.02  2923.2  910.46  3054.4   909.9
  3291.6  909.13  3352.5  903.64  3408.2  909.14  3436.9  909.51  3687.4  911.66
  3949.1  921.44  4086.7  914.63    4118  908.22  4199.5  908.04  4243.5  903.71
  4357.5  902.25  4377.5  907.99  4440.9  909.38  4955.3  908.78  4969.1  903.68
  4974.6  903.48  4978.5   895.2  4981.5   894.6  5009.5   895.2  5022.4  895.65
  5055.3  909.85    5093  907.52  5846.5  909.63  6253.5  926.79  6600.9  936.35
#Mann= 11 ,-1 , 0
  1834.8     .05       0    2547     .05       0  2824.4     .05       0
  2923.2     .05       0  3054.4     .05       0  3408.2     .05       0
  3436.9     .05       0  4969.1     .16       0  4978.5     .07       0
  5009.5     .16       0    5093     .05       0
#XS Ineff= 2 , 0
       0  3934.6  928.37               0
Permanent Ineff=
       F       F
Bank Sta=4978.5,5009.5
XS Rating Curve= 0 ,0
Exp/Cntr=0.3,0.1

Type RM Length L Ch R = 1 ,492109  ,932,932,932
BEGIN DESCRIPTION:
Denton Creek 214.0
END DESCRIPTION:
XS GIS Cut Line= 3
      2221268.32      7240585.05        2219179.        7237960.
      2218934.95       7237225.4
#Sta/Elev= 30
  1657.4  935.57  2117.9  916.66  2143.8  915.86  2456.2  906.49  2879.6  905.91
  2914.8  905.81  3010.4  906.09  3050.1  905.98  3348.5   906.2  3476.7   906.3
  4236.4  910.54  4335.7  897.77  4386.2  897.07  4414.2  907.21    4443  908.52
  4926.7  906.68  4976.4  900.07  4992.2  891.19  4994.4  891.05  5001.8  890.59
  5011.4  891.19  5028.3  911.15    5044  914.32  5091.6  904.38  5126.6  905.05
  5222.7  911.56  5482.5  929.18  5546.5  932.69  5624.6  937.98  5786.5  946.62
#Mann= 18 ,-1 , 0
  1657.4     .05       0  2117.9     .05       0  2143.8     .05       0
  2456.2     .05       0  2879.6     .05       0  2914.8     .05       0
  3010.4     .05       0  3050.1     .05       0  3348.5     .05       0
  3476.7     .05       0  4992.2     .07       0  4994.4     .16       0
  5011.4     .05       0  5126.6     .05       0  5222.7     .16       0
  5482.5     .05       0  5546.5     .16       0  5624.6     .05       0
#XS Ineff= 2 , 0
       0  4236.8  928.51               0
Permanent Ineff=
       F       F
Bank Sta=4992.2,5011.4
XS Rating Curve= 0 ,0
Exp/Cntr=0.3,0.1

Type RM Length L Ch R = 1 ,491177  ,820,820,820
BEGIN DESCRIPTION:
Denton Creek 213.0
END DESCRIPTION:
XS GIS Cut Line= 3
      2222154.45      7239480.93        2220029.        7237660.
      2218973.05      7236718.55
#Sta/Elev= 30
  2207.8     961  2411.3  949.03  2510.1  939.34  2840.8  916.72  2949.4  909.73
  3112.7  902.29  3755.6  903.95  4021.7  905.24  4602.1   905.3  4743.9  907.83
  4942.4  907.18  4956.7  900.18  4978.6   894.9  4982.4  890.75  4987.2  889.75
  5024.2  890.75  5027.9     897    5063   907.4  5132.4  908.32    5191  903.99
  5233.6  905.95  5297.1  913.62  5342.6  912.88  5488.6  912.24  5759.1  924.13
  5762.6  924.35  6019.5  932.83  6084.6  931.82  6217.7  932.74  6421.3  944.59
#Mann= 13 ,-1 , 0
  2207.8     .05       0  2840.8     .05       0  2949.4     .05       0
  3755.6     .05       0  4021.7     .05       0  4743.9     .05       0
  4982.4    .035       0  5024.2     .05       0  5132.4     .05       0
  5342.6     .16       0  5759.1     .05       0  5762.6     .16       0
  6084.6     .05       0
#XS Ineff= 2 , 0
       0    4673  932.14               0
Permanent Ineff=
       F       F
Bank Sta=4982.4,5024.2
XS Rating Curve= 0 ,0
Exp/Cntr=0.3,0.1

Type RM Length L Ch R = 1 ,490357  ,975,975,975
BEGIN DESCRIPTION:
Denton Creek 212.0
END DESCRIPTION:
XS GIS Cut Line= 3
      2222310.74      7238212.31      2220517.55       7237166.4
      2218922.18      7236543.47
#Sta/Elev= 30
  3137.9  931.22  3315.3  927.41  3370.1  917.23  3395.5  916.35  3432.7  921.94
  3534.4  922.01  3834.5  910.28  4019.7  915.77  4223.3  903.01  4377.9  899.85
  4900.9  906.54    4969  906.49  4976.6  903.22  4977.2  889.53    4982  888.53
    5019  889.53  5019.6  894.47  5072.7  897.82  5099.8  905.62  5137.1  907.45
  5195.8  908.95    5223  905.77    5309  905.53  5530.9  904.39  5573.5  902.58
  5820.7  908.74    6411   915.8  6537.7   919.1  6839.2  936.66  6926.5   938.4
#Mann= 9 ,-1 , 0
  3137.9     .05       0  3370.1     .05       0  4900.9     .05       0
  4977.2    .035       0    5019     .05       0  5072.7     .16       0
    5309     .05       0  5530.9     .16       0    6411     .05       0
Bank Sta=4977.2,5019
XS Rating Curve= 0 ,0
Exp/Cntr=0.3,0.1

Type RM Length L Ch R = 1 ,489382  ,1583,1583,1583
BEGIN DESCRIPTION:
Denton Creek 211.0
END DESCRIPTION:
XS GIS Cut Line= 3
      2222079.03      7237410.03        2221079.        7236410.
      2219313.56      7234865.42
#Sta/Elev= 30
  3578.2  930.81  4059.1  899.61  4098.2  898.66  4210.4  900.81  4271.2  898.73
  4299.5  901.07  4402.8  900.19  4704.5  901.33  4877.8  903.37    4950  903.17
  4985.3  888.52  4990.1  887.52  5027.1  888.52  5028.1  893.09  5034.7  894.04
  5042.3  899.19  5056.5   904.8  5276.6  901.76  5367.8  902.29  5424.8  899.29
  5445.7  901.88  5573.8  901.09  5602.3  898.64  5651.6  900.34  6100.8  900.34
  6735.5  905.32  6973.2  912.35    7211  925.23  7231.9  929.36  7338.2  937.17
#Mann= 11 ,-1 , 0
  3578.2     .05       0  4098.2     .05       0  4210.4     .05       0
  4402.8     .05       0  4704.5     .05       0  4877.8     .05       0
  4985.3     .07       0  5027.1     .16       0  5276.6     .16       0
  6100.8     .05       0  6973.2     .05       0
Bank Sta=4985.3,5027.1
XS Rating Curve= 0 ,0
Exp/Cntr=0.3,0.1

Type RM Length L Ch R = 1 ,487799  ,1189,1189,1189
BEGIN DESCRIPTION:
Denton Creek 209.0
END DESCRIPTION:
XS GIS Cut Line= 3
      2223199.49       7236624.1      2222026.48       7235329.1
      2220326.35      7233418.88
#Sta/Elev= 30
  3090.2  920.96  3383.6   903.4  3624.2   898.4  4176.4  895.58  4927.4  903.24
  4948.3  901.12  4962.5  891.65  4976.5  886.56  4981.3  885.56  5018.7  886.56
  5019.3  890.35  5045.9  897.13    5059  901.48  5326.8  900.75  5333.1  900.98
  5480.6  900.23  5594.6  900.02  5625.5  900.42  5728.5  901.06  6130.1  902.83
  6205.2   903.3  6275.5  903.71  6388.4  903.87  6690.8  905.04  6995.2  913.19
  7137.3  913.91  7166.9  910.88  7229.3  909.02    7272  918.19  7394.7   924.8
#Mann= 16 ,-1 , 0
  3090.2     .05       0  4976.5     .05       0  5018.7     .05       0
  5045.9     .05       0    5059     .05       0  5326.8     .05       0
  5333.1     .05       0  5480.6     .05       0  5594.6     .05       0
  5625.5     .05       0  5728.5     .05       0  6130.1     .05       0
  6205.2     .05       0  6275.5     .05       0  6388.4     .05       0
  7166.9     .05       0
Bank Sta=4976.5,5018.7
XS Rating Curve= 0 ,0
Exp/Cntr=0.3,0.1

Type RM Length L Ch R = 1 ,486610  ,949,949,949
BEGIN DESCRIPTION:
Denton Creek 208.0
END DESCRIPTION:
XS GIS Cut Line= 3
      2224093.04      7236282.03        2222629.        7234310.
      2222129.02      7233410.04
#Sta/Elev= 30
  2515.8  924.47  2750.6  924.25  2792.3  917.41    2881  916.92  3084.8  905.76
  3671.1  895.82  4372.1  893.94  4745.4  898.39  4848.4  899.74  4857.1  899.68
    4950   897.9  4958.3  890.72  4985.9  885.11  4990.6  884.11  5028.7  885.11
  5029.1  888.33  5088.6  899.17    5132  899.26  5142.3  894.91    5148  897.36
  5154.9  890.93  5162.4  888.99  5191.5  888.72  5207.5  899.08  5230.2   900.4
  5419.2  897.35  5559.9  899.29  5722.3  906.55  5852.7  920.33  6001.4  925.87
#Mann= 10 ,-1 , 0
  2515.8     .16       0  2750.6     .05       0    2881     .05       0
  4745.4     .05       0  4848.4     .05       0  4857.1     .05       0
  4985.9    .035       0  5028.7     .05       0  5162.4     .16       0
  5230.2     .05       0
Bank Sta=4985.9,5028.7
XS Rating Curve= 0 ,0
Exp/Cntr=0.3,0.1

Type RM Length L Ch R = 1 ,485661  ,960,960,960
BEGIN DESCRIPTION:
Denton Creek 207.0
END DESCRIPTION:
XS GIS Cut Line= 3
      2224580.51      7236008.14        2223179.        7233660.
        2223079.        7233160.
#Sta/Elev= 30
  2256.5  938.34  2384.1  929.41  2439.8  925.35  2461.2     921    2512  921.46
    2627  913.54  2673.4   907.8  2700.6  909.75    2759   904.6  2827.7  902.23
  3008.1  897.56  3517.9  892.56  3896.8  893.65  4250.9  895.52  4366.3  896.84
  4558.4  895.77  4874.6  897.62  4924.9  899.62  4932.9  898.81  4940.5  894.16
  4946.3  895.04  4961.9  891.03  4966.6  883.46  4971.3  882.46  5009.7  883.46
  5031.9  888.35  5055.4  897.07  5072.7  899.17  5154.3  899.29    5501  920.76
#Mann= 11 ,-1 , 0
  2256.5     .05       0  2384.1     .16       0    2512     .05       0
  2827.7     .05       0  3896.8     .12       0  4250.9     .05       0
  4366.3     .05       0  4558.4     .05       0  4966.6    .035       0
  5009.7     .05       0  5055.4     .05       0
Bank Sta=4966.6,5009.7
XS Rating Curve= 0 ,0
Exp/Cntr=0.3,0.1

Type RM Length L Ch R = 1 ,484701  ,1897,1897,1897
BEGIN DESCRIPTION:
Denton Creek 206.0
END DESCRIPTION:
XS GIS Cut Line= 3
      2226303.59      7235021.96        2223879.        7233160.
      2223233.12      7232665.65
#Sta/Elev= 30
  1930.6  934.24    2285  918.65  2376.8  910.88  2598.6  905.75  2648.4  900.28
  2762.6  895.78  2828.4  897.66  2850.3  897.57  3005.5  894.27  3375.2  892.24
  4074.6  891.37  4320.6  892.49  4322.1  892.43  4443.7  893.02  4568.6  893.49
  4791.8  896.67  4945.1  896.62  4951.4  891.38  4974.1  886.23  4979.7  882.31
  4984.4  881.31  5022.8  882.31    5024  891.04  5051.1  897.45  5188.1  894.88
  5301.4  897.47  5543.4  905.29  5593.3  909.01  5791.1  911.87    5801  912.34
#Mann= 14 ,-1 , 0
  1930.6     .05       0  2376.8     .05       0  2828.4     .05       0
  2850.3     .05       0  4074.6     .05       0  4320.6     .05       0
  4322.1     .05       0  4443.7     .05       0  4568.6     .05       0
  4791.8     .05       0  4979.7    .035       0  5022.8     .05       0
  5301.4     .05       0  5791.1     .05       0
Bank Sta=4979.7,5022.8
XS Rating Curve= 0 ,0
Exp/Cntr=0.3,0.1

Type RM Length L Ch R = 1 ,482804  ,797,797,797
BEGIN DESCRIPTION:
Denton Creek 204.0
END DESCRIPTION:
XS GIS Cut Line= 4
      2226139.29      7233139.72      2225557.67      7232706.45
      2225307.33      7232418.72      2223740.02      7231366.52
#Sta/Elev= 30
  4096.8  923.33  4236.9  912.63  4260.4  908.48  4289.6  909.64  4304.2  906.84
  4325.1  910.18  4574.9  895.94  4696.3  892.87    4859  893.43  4960.7  889.41
  4981.3  879.26  4985.9  878.26  5024.6  879.26  5030.9  885.97  5038.5   887.8
  5059.4  888.72  5081.2     885  5102.1  891.34  5144.9  892.42  5165.7  889.89
  5194.2  890.39  5214.8  894.23  5259.5  893.69    6247  892.99  6844.1  904.32
  6916.2  907.21  6931.1  911.22  6952.2  907.43  7060.2  916.86  7091.2  916.17
#Mann= 7 ,-1 , 0
  4096.8     .05       0  4236.9     .05       0  4574.9     .05       0
    4859     .05       0  4981.3    .035       0  5024.6     .05       0
  5259.5     .05       0
Bank Sta=4981.3,5024.6
XS Rating Curve= 0 ,0
Exp/Cntr=0.3,0.1

Type RM Length L Ch R = 1 ,482007  ,216,216,216
BEGIN DESCRIPTION:
Denton Creek292
END DESCRIPTION:
XS GIS Cut Line= 3
      2226828.85      7232542.06      2225617.87      7231833.91
      2223865.03      7230804.51
#Sta/Elev= 30
  3996.3  926.36  4158.3  915.67  4239.4  916.62    4488  903.99  4578.5  899.48
    4585   899.2  4700.3  893.46  4932.3  891.64  4940.8  886.31  4969.2  884.38
  4977.7   878.5  4982.4   877.5  5021.2   878.5  5027.1  884.35  5032.5  885.27
  5079.6  893.43  5145.6  893.47  5282.9  890.42  5325.2  892.94  5606.5  890.79
    6424  891.27  6673.5  899.59  6754.2  910.33  6818.6   903.3  6877.2  903.04
  6941.6  912.41  7067.8  920.61  7154.6  925.38  7264.9  924.82  7431.9  934.48
#Mann= 11 ,-1 , 0
  3996.3     .05       0    4488     .05       0  4578.5     .05       0
    4585     .05       0  4932.3     .05       0  4977.7    .035       0
  5021.2     .05       0  5032.5     .05       0  5145.6     .05       0
  5325.2     .05       0  5606.5     .05       0
Bank Sta=4977.7,5021.2
XS Rating Curve= 0 ,0
Exp/Cntr=0.3,0.1

Type RM Length L Ch R = 1 ,481791  ,854,854,854
BEGIN DESCRIPTION:
Denton Creek 203.0
END DESCRIPTION:
XS GIS Cut Line= 3
      2226916.09      7232447.56      2226341.12      7232014.33
      2223965.22      7230638.14
#Sta/Elev= 30
  4008.2  928.42    4276  913.96  4296.9  917.94  4311.4   914.1  4317.7  917.86
  4355.1  917.42  4675.8  894.88  4902.2  894.49  4923.8  886.69  4961.1  886.96
  4973.2  883.01  4974.6  877.89  4979.3  876.89  5018.1  877.89  5019.5  883.31
  5025.6  886.54  5076.2  889.89    5135  893.67  5472.1  891.38  5971.3   889.3
  6319.9  889.48  6545.7  891.44  6658.6  894.83  6693.4  897.87  6840.6  913.79
  6884.3  912.16  7065.9  909.43  7183.5  921.01  7335.9  926.64  7473.8  931.87
#Mann= 12 ,-1 , 0
  4008.2     .05       0  4974.6    .035       0  5018.1     .05       0
  5076.2     .05       0  5472.1     .05       0  5971.3     .16       0
  6319.9     .05       0  6545.7     .05       0  6658.6     .05       0
  6693.4     .05       0  6884.3     .05       0  7335.9    .063       0
Bank Sta=4974.6,5018.1
XS Rating Curve= 0 ,0
Exp/Cntr=0.3,0.1

Type RM Length L Ch R = 1 ,480937  ,1376,1376,1376
BEGIN DESCRIPTION:
Denton Creek 202.0
END DESCRIPTION:
XS GIS Cut Line= 3
      2227129.01      7232310.02        2226729.        7231310.
      2225328.97      7229909.97
#Sta/Elev= 30
  3905.6  935.78  4060.7  925.88  4379.8   908.2  4488.6  898.04  4620.5  890.92
  4767.2   889.7  4806.3  892.83  4878.7   892.2  4943.6  892.45  4961.1   887.8
  4973.2  880.54    4975  877.28  4979.7  876.28  5018.5  877.28  5025.1  881.76
  5029.8  882.35  5095.8  893.79  5124.1   889.6  5171.6  889.49  6099.9  888.83
  6223.9   886.5  6288.4  885.91  6467.6  885.82  6538.3  889.53  6566.6  895.37
  6590.1  894.87  6599.9   894.7  6722.1  903.07  6920.1  920.22  6962.6  921.64
#Mann= 12 ,-1 , 0
  3905.6     .05       0  4060.7     .16       0  4379.8     .05       0
  4878.7     .16       0    4975     .07       0  5018.5     .16       0
  5029.8     .05       0  5171.6     .05       0  6223.9     .05       0
  6288.4     .05       0  6590.1     .05       0  6599.9     .05       0
Bank Sta=4975,5018.5
XS Rating Curve= 0 ,0
Exp/Cntr=0.3,0.1

Type RM Length L Ch R = 1 ,479561  ,1783,1783,1783
BEGIN DESCRIPTION:
Denton Creek 200.0
END DESCRIPTION:
XS GIS Cut Line= 3
      2228922.19      7232072.05      2227631.05      7230286.64
      2224964.06      7228187.25
#Sta/Elev= 30
  2628.6  927.25  2774.5  925.66  2983.4  920.57  3261.8  904.29  3356.2  908.08
  3412.6  901.95  3462.9  905.98  3619.9  895.45  3655.5  898.21  3714.3  892.32
  4606.6  886.01  4777.4  887.23  4914.3  889.72  4935.2  891.94  4959.7  888.46
  4979.6   876.2  4984.2   875.2  5023.1   876.2  5023.8  881.26    5038  883.36
  5123.3  887.98  6505.2  886.21  6645.5  886.81  6769.2  887.44  6803.9  893.66
  6967.5     891  7565.6  926.93  7878.3   930.4  8000.2  936.64  8226.1  927.92
#Mann= 12 ,-1 , 0
  2628.6     .05       0  2774.5     .05       0  4606.6     .16       0
  4777.4     .05       0  4914.3     .16       0  4935.2     .05       0
  4979.6    .035       0  5023.1     .05       0    5038     .05       0
  6505.2     .05       0  6645.5     .05       0  6769.2     .05       0
Bank Sta=4979.6,5023.1
XS Rating Curve= 0 ,0
Exp/Cntr=0.3,0.1

Type RM Length L Ch R = 1 ,477778  ,2329,2329,2329
BEGIN DESCRIPTION:
Denton Creek 198.0
END DESCRIPTION:
XS GIS Cut Line= 3
      2230208.16       7230026.2      2227054.17      7227619.64
      2225019.49      7228057.83
#Sta/Elev= 30
  2877.2  942.81  3052.2  937.85  3123.9  924.65  3180.1  927.83  3252.8  917.33
  3358.8   922.6  3872.2     924  4244.2  900.16  4300.4  907.02    4344  896.24
  4707.7  885.72  4736.7  876.41  4750.3  884.07  4839.6  888.74  4936.3  889.65
  4964.2  879.83  4964.4  874.21    4969  873.21    5008  874.21  5048.4  890.46
  5270.5  886.39  5761.3  886.37  6654.6  889.68  6754.9  894.47    6784  889.01
  6893.3  890.97    7982  895.28    8293  897.88  8619.1  912.67  8925.8   922.1
#Mann= 12 ,-1 , 0
  2877.2     .05       0  4839.6     .16       0  4964.4     .07       0
    5008     .16       0  5048.4     .05       0  5270.5     .16       0
  5761.3     .05       0  6654.6     .05       0  6893.3     .05       0
    7982     .05       0    8293     .16       0  8619.1     .05       0
Bank Sta=4964.4,5008
XS Rating Curve= 0 ,0
Exp/Cntr=0.3,0.1

Type RM Length L Ch R = 1 ,475449  ,1168,1168,1168
BEGIN DESCRIPTION:
Denton Creek 196.0
END DESCRIPTION:
XS GIS Cut Line= 3
      2230769.53       7227909.6        2229879.        7226860.
      2226434.66      7223480.48
#Sta/Elev= 30
  3648.5  929.16  3715.3  925.21  3840.3  919.14  4067.6  923.04  4119.3  919.19
    4280  908.62    4316  902.64  4351.1  906.75  4357.7   903.3  4379.7  905.86
  4492.7  898.92  4592.2  899.85  4620.2  893.31    4684   890.2  4857.9  887.22
  4946.4  887.99  4993.8  871.95    4998  870.95  5041.9  871.95  5046.2  886.24
  5060.3     888  5901.8  880.44  6315.1  881.07  6441.2  881.97  7092.8  882.22
  7726.3  882.46  8588.9  890.04  9089.6  906.03  9303.2   916.1  9850.4  953.37
#Mann= 12 ,-1 , 0
  3648.5     .05       0  3715.3     .16       0  4119.3     .05       0
    4280     .16       0  4492.7     .05       0  4857.9     .16       0
  4993.8     .07       0  5041.9     .16       0  6315.1     .12       0
  6441.2     .05       0  7092.8     .05       0  9089.6     .16       0
#XS Ineff= 2 , 0
       0                    6800       0     918
Permanent Ineff=
       F       F
Bank Sta=4993.8,5041.9
XS Rating Curve= 0 ,0
Exp/Cntr=0.3,0.1

Type RM Length L Ch R = 1 ,474281  ,1717,1717,1717
BEGIN DESCRIPTION:
Denton Creek 194.0
END DESCRIPTION:
XS GIS Cut Line= 3
       2231149.8      7227977.61       2230936.4      7226577.62
      2229564.62       7222273.5
#Sta/Elev= 30
  3133.2  932.59    3361  930.34  3531.2  920.98  4035.3  894.12  4181.9  892.14
    4363  888.42  4385.1  894.43  4436.7  886.06  4636.6  882.92  4847.9   885.3
  4935.2  886.92  4963.7  878.86  4989.2  876.73  4992.1  870.83  4996.3  869.83
  5040.2  870.83  5071.6  886.74  5134.6  886.96    6541  876.01  7258.8  877.12
  7422.9  877.52  7695.6  881.45    7727  887.45  7778.8  878.13  7842.5  877.14
  8079.8  896.51  8296.2  903.81  8650.9  928.65  8844.1  941.65  9066.8  957.57
#Mann= 15 ,-1 , 0
  3133.2     .05       0    3361     .05       0  3531.2     .16       0
  4181.9     .05       0  4636.6     .05       0  4847.9     .05       0
  4963.7     .16       0  4992.1     .07       0  5040.2     .16       0
  7258.8     .05       0  7422.9     .16       0  7778.8     .05       0
  8296.2     .16       0  8650.9     .05       0  8844.1     .16       0
Bank Sta=4992.1,5040.2
XS Rating Curve= 0 ,0
Exp/Cntr=0.3,0.1

Type RM Length L Ch R = 1 ,472564  ,2042,2042,2042
BEGIN DESCRIPTION:
Denton Creek 193.0
END DESCRIPTION:
XS GIS Cut Line= 3
      2232199.58      7227523.11      2232229.48      7226006.43
      2231517.24      7221574.77
#Sta/Elev= 30
  2485.7     910  2578.8  904.92  2608.8  897.14  2658.8  900.02  2847.1  890.55
  3235.8  882.79  3668.1  880.73    3677  880.73  3774.7  881.06  4168.5  881.56
  4267.9  882.31  4777.2   883.9  4917.6  885.57  4953.9  881.17  4961.2  879.15
  4967.5  869.23  4971.7  868.23  5015.8  869.23  5133.4  884.31  5942.1  875.52
  6288.1  877.04    6681  904.62    7057  908.91  7233.5  912.73  7260.4  905.18
  7300.9  914.97    7611  921.62  8131.7  947.56  8344.4  959.78  8491.2     959
#Mann= 19 ,-1 , 0
  2485.7     .05       0  2847.1     .05       0  3235.8     .05       0
  3668.1     .05       0    3677     .05       0  3774.7     .05       0
  4168.5     .05       0  4267.9     .05       0  4777.2     .05       0
  4953.9     .16       0  4967.5     .07       0  5015.8     .16       0
  5942.1     .05       0  6288.1     .16       0    7057     .05       0
  7233.5     .16       0    7611     .05       0  8131.7    .063       0
  8344.4     .16       0
Bank Sta=4967.5,5015.8
XS Rating Curve= 0 ,0
Exp/Cntr=0.3,0.1

Type RM Length L Ch R = 1 ,470522  ,1583,1583,1583
BEGIN DESCRIPTION:
Denton Creek 191.0
END DESCRIPTION:
XS GIS Cut Line= 3
      2235138.22      7227963.02      2234190.05      7224734.32
      2232731.42      7222145.62
#Sta/Elev= 30
   628.1  905.99  1099.7  911.42  1558.8  894.28  1669.1  885.67    1901  876.16
  2418.2     876  2490.5  876.23  2879.4  876.75    3094  881.49  3252.2  878.96
  4973.6  879.78  4981.4  874.88  4983.8  866.57  4987.8  865.57  5033.8  866.57
  5040.6   874.2    5084  877.42  5208.2  877.99  5283.4  869.45  5326.7  871.65
  5354.1  882.04  5618.5  883.62  5788.7  896.96  5898.8   900.8  5958.1  895.56
  5979.7  903.69  6086.6  905.84    6263  908.15  6569.2  919.48  6964.5  940.34
#Mann= 14 ,-1 , 0
   628.1     .16       0  1669.1     .05       0    1901     .05       0
  2418.2     .05       0  2490.5     .05       0  2879.4     .16       0
  3252.2     .05       0  4973.6     .16       0  4983.8     .07       0
  5033.8     .16       0  5979.7     .05       0  6086.6     .16       0
    6263     .05       0  6569.2     .16       0
#XS Ineff= 2 , 0
       0  3190.9  913.88               0
Permanent Ineff=
       F       F
Bank Sta=4983.8,5033.8
XS Rating Curve= 0 ,0
Exp/Cntr=0.3,0.1

Type RM Length L Ch R = 1 ,468939  ,1864,1864,1864
BEGIN DESCRIPTION:
Denton Creek 190.0
END DESCRIPTION:
XS GIS Cut Line= 3
      2237950.23       7226885.2      2234624.81      7222701.57
       2234024.2      7221636.86
#Sta/Elev= 30
     271  945.24   987.4  914.65  1990.2  896.11  2147.2  883.74  2318.6  886.86
    2389  882.26  2567.7  883.88  2645.4   887.9  2909.1  872.09  3205.5  873.66
  4572.2  879.16  4944.1  881.15    4973  876.75  4976.8  864.89  4980.8  863.89
  5026.8  864.89  5043.4  872.74  5128.2  875.14  5250.1  874.32  5264.5  880.86
    5296  884.57    5505  879.99  5570.5  878.94  5679.1  887.67  5810.7  890.59
  5869.8  893.45    6012   904.1  6126.9  912.91  6434.5  925.36  6837.7  933.17
#Mann= 12 ,-1 , 0
     271     .16       0  2567.7     .05       0  3205.5     .05       0
  4572.2     .05       0  4976.8     .07       0  5026.8     .05       0
  5128.2     .05       0    5296     .16       0    5505     .05       0
  5810.7     .16       0  5869.8     .05       0    6012     .16       0
Bank Sta=4976.8,5026.8
XS Rating Curve= 0 ,0
Exp/Cntr=0.3,0.1

Type RM Length L Ch R = 1 ,467075  ,1333,1333,1333
BEGIN DESCRIPTION:
Denton Creek 189.0
END DESCRIPTION:
XS GIS Cut Line= 3
      2238801.48      7225043.02        2236329.        7222160.
       2235582.1      7220694.47
#Sta/Elev= 30
    1195  911.36  1203.3  911.06  1454.1  904.39    1532  896.99  1546.3  899.42
  2080.9  885.56  2238.9  880.02  3453.7  871.44    4754  876.48  4782.2   877.4
  4928.8  877.24  4979.3  869.61  4981.9  860.92  4985.9  859.92  5031.9  860.92
  5037.9   868.7  5140.4   876.5  5172.6  872.85  5179.2  875.34  5184.8  871.22
  5223.7  878.33  5290.4  878.13  5329.2  883.32    5396  881.71  5632.8  892.79
  5798.4  892.89  6079.6  900.56  6253.3  912.51  6390.9  920.49  6637.9  925.32
#Mann= 10 ,-1 , 0
    1195     .05       0  1203.3     .16       0  2080.9     .05       0
  2238.9     .16       0    4754     .05       0  4782.2     .16       0
  4981.9     .07       0  5031.9     .16       0  5798.4     .05       0
  6253.3     .16       0
Bank Sta=4981.9,5031.9
XS Rating Curve= 0 ,0
Exp/Cntr=0.3,0.1

Type RM Length L Ch R = 1 ,465742  ,1409,1409,1409
BEGIN DESCRIPTION:
Denton Creek 188.0
END DESCRIPTION:
XS GIS Cut Line= 3
      2239651.92      7223304.74        2237379.        7221360.
      2235567.56      7220319.83
#Sta/Elev= 30
  1998.8  927.95  2394.6   905.8  2792.4  877.97  2907.9  873.32  3412.2  870.72
  3418.5  870.57  3536.2  870.72  3593.3  866.75  3663.6   871.9  4132.3  872.46
    4196  869.92  4805.9  874.22  4865.1  871.83    4944  867.99  4976.4  867.07
  4978.8  858.54  4982.8  857.54  5028.8  858.54  5035.4  868.89    5063  873.71
  6097.2  875.39  6293.2  885.16  6404.3  896.76  6484.9  900.98  6543.8  899.89
  6571.1  895.55  6726.4  908.52    6852  907.34  6960.6  911.35    7079  911.42
#Mann= 12 ,-1 , 0
  1998.8     .16       0  2792.4     .05       0  2907.9     .16       0
  3412.2     .05       0  3418.5     .16       0  4865.1     .05       0
    4944     .16       0  4978.8     .07       0  5028.8     .16       0
    5063     .05       0    6852     .16       0  6960.6     .05       0
Bank Sta=4978.8,5028.8
XS Rating Curve= 0 ,0
Exp/Cntr=0.3,0.1

Type RM Length L Ch R = 1 ,464333  ,1378,1378,1378
BEGIN DESCRIPTION:
Denton Creek 187.0
END DESCRIPTION:
XS GIS Cut Line= 3
      2241803.99      7222097.09        2238329.        7220360.
        2236529.        7218760.
#Sta/Elev= 30
  1146.1  928.84  1421.7  916.96  1511.8  912.36  1528.6  900.68    1543   909.4
  1656.2  902.36  1859.4  892.66  1886.4  891.04  1968.8  888.77  2316.9  887.18
  2445.4  875.51  2515.9  879.64    2606  876.63    3063  870.41  3802.5   867.9
  4770.3  868.51    4964  870.88  4972.4  870.19  4975.3  855.53  4979.3  854.53
  5025.3  855.53  5028.3  865.74  5065.7  866.23  5087.5  870.75  5215.5  871.71
  6568.5  873.16  6979.5  909.65  7177.2  928.25    7439  933.58  7439.4  933.58
#Mann= 16 ,-1 , 0
  1146.1     .05       0  1421.7     .16       0  1656.2     .05       0
  1859.4     .16       0  1886.4     .05       0  1968.8     .16       0
  2515.9     .05       0    2606     .05       0    3063     .05       0
  3802.5     .16       0  4770.3     .05       0  4975.3     .07       0
  5025.3     .05       0  5065.7     .05       0  6979.5     .16       0
    7439     .05       0
Bank Sta=4975.3,5025.3
XS Rating Curve= 0 ,0
Exp/Cntr=0.3,0.1

Type RM Length L Ch R = 1 ,462955  ,2155,2155,2155
BEGIN DESCRIPTION:
Denton Creek 186.0
END DESCRIPTION:
XS GIS Cut Line= 3
      2241635.27      7219415.13        2238929.        7219160.
       2236232.5       7218040.3
#Sta/Elev= 30
  2289.2  920.87  2657.1  917.29  2981.7  903.21    3394  889.05  3552.1  890.73
    3692  886.26  3842.3  874.95  4093.4  863.27  4545.6  866.66  4760.5  867.13
  4958.2  870.52  4967.3  869.53  4972.4  854.08  4976.4  853.08  5022.4  854.08
  5023.3  856.32  5029.1  870.77  5475.2   867.8  5678.8  868.33  5702.2   865.5
  5755.3  868.89  6459.3   868.6  6642.3  879.67  6750.8  882.68  7157.8  913.56
  7553.7  916.37  7668.1  922.95  7746.9  930.73  7790.2   940.5  7927.2  938.14
#Mann= 13 ,-1 , 0
  2289.2     .05       0  2981.7     .16       0    3394     .05       0
  3552.1     .16       0    3692     .05       0  4545.6     .16       0
  4760.5     .05       0  4972.4    .035       0  5022.4     .05       0
  5023.3     .16       0  5475.2     .05       0  6642.3     .16       0
  7668.1     .05       0
Bank Sta=4972.4,5022.4
XS Rating Curve= 0 ,0
Exp/Cntr=0.3,0.1

Type RM Length L Ch R = 1 ,460800  ,3197,3197,3197
BEGIN DESCRIPTION:
Denton Creek 185.0
END DESCRIPTION:
XS GIS Cut Line= 4
      2242250.44      7218755.45      2239442.45      7217193.92
      2238728.99      7217125.56      2235959.89       7217123.1
#Sta/Elev= 30
  1462.8  923.57  1710.5  922.09  1894.7  902.83  1954.1  902.51  1990.8  916.87
  2041.1  916.35  2093.8  902.61    2144  915.09  2219.5  916.24  2393.3  910.36
  2447.1  898.06    2550  911.72  2658.6  914.13  2859.9  901.75  3427.5  868.07
  4506.6  864.16  4960.5  864.81  4970.6  863.06  4975.7  852.67  4979.7  851.67
  5025.7  852.67  5030.8  864.41  5157.9  860.97  5282.6  862.88  5644.1  884.87
  6162.5  871.89  6541.9  881.69    6945  881.05  7806.7  918.91  8161.6  939.11
#Mann= 12 ,-1 , 0
  1462.8     .05       0  2859.9     .16       0  3427.5     .05       0
  4506.6     .16       0  4975.7     .07       0  5025.7     .16       0
  5157.9     .16       0  5282.6     .05       0  5644.1     .16       0
  6541.9     .05       0    6945     .16       0  7806.7     .05       0
Bank Sta=4975.7,5025.7
XS Rating Curve= 0 ,0
Exp/Cntr=0.3,0.1

Type RM Length L Ch R = 1 ,457603  ,391,391,391
BEGIN DESCRIPTION:
Denton Creek291
END DESCRIPTION:
XS GIS Cut Line= 4
      2241705.25       7217337.8        2240738.      7216394.52
      2237991.41      7213711.58      2237644.32      7213604.87
#Sta/Elev= 30
   658.3  912.03   746.1  905.81  1124.6  891.08  1318.9  880.77  1516.9  874.13
  1644.2  865.97  2183.7  858.92  3143.9  859.19  3181.9   859.2  3265.1  859.22
  3325.5  859.48  3400.3  859.61  3469.1  858.78  3535.5  859.27  3590.1  859.23
  4430.1  859.49    4617  860.35  4711.7  860.01  4865.5  860.11  4960.6   858.9
  4974.8  855.95  4978.1  849.31  4982.1  848.31  5028.1  849.31  5031.4  855.71
  5045.5  860.21  5257.7  858.28  5494.4  862.81    5877  882.52    6212  898.93
#Mann= 20 ,-1 , 0
   658.3     .05       0  1124.6     .16       0  1318.9     .05       0
  2183.7     .05       0  3143.9     .05       0  3181.9     .05       0
  3265.1     .05       0  3325.5     .05       0  3400.3     .05       0
  3469.1     .05       0  3535.5     .05       0  3590.1     .05       0
  4430.1     .05       0    4617     .05       0  4711.7     .05       0
  4865.5     .05       0  4978.1    .045       0  5028.1     .05       0
  5494.4     .05       0    5877     .16       0
Bank Sta=4978.1,5028.1
XS Rating Curve= 0 ,0
Exp/Cntr=0.3,0.1

Type RM Length L Ch R = 1 ,457212  ,1358,1358,1358
BEGIN DESCRIPTION:
Denton Creek 182.0
END DESCRIPTION:
XS GIS Cut Line= 3
      2241880.32      7217235.44      2238271.47       7213547.7
      2237784.49      7213460.49
#Sta/Elev= 30
   371.2  915.91   651.8  911.65   694.2  905.55   729.5  907.39   998.2  892.82
    1066  891.51  1528.6  872.62    1980  861.05  2297.9  859.68  4350.7  860.88
  4393.3  860.92  4795.7  861.07  4816.8  864.72  4866.4  865.31  4965.4  859.39
  4975.7  848.52  4979.7  847.52  5025.7  848.52  5043.1  856.84  5085.6  861.21
  5191.7  857.61  5297.7  859.22  5509.9  866.31  5624.9  875.66    5655  871.21
  5726.5   874.5    5757  885.49  5802.9   889.7    5950   899.2  6025.7  898.94
#Mann= 10 ,-1 , 0
   371.2     .05       0   998.2     .16       0    1066     .05       0
    1980     .05       0  2297.9     .05       0  4350.7     .05       0
  4393.3     .05       0  4975.7    .035       0  5025.7     .05       0
  5802.9     .16       0
Bank Sta=4975.7,5025.7
XS Rating Curve= 0 ,0
Exp/Cntr=0.3,0.1

Type RM Length L Ch R = 1 ,455854  ,2479,2479,2479
BEGIN DESCRIPTION:
Denton Creek 181.0
END DESCRIPTION:
XS GIS Cut Line= 3
      2241982.26      7215490.84      2240658.22      7213484.77
      2237571.17      7212004.57
#Sta/Elev= 30
   601.5  890.86   792.2  883.67   911.3  876.52  1211.6  866.36    2018  865.07
  2423.7  865.72  2792.1  858.74  2813.1   862.7    3359  860.78  4926.4  859.77
  4943.5  863.46  4971.7  855.06  4975.5  846.48  4979.5  845.48  5025.5  846.48
  5033.8  860.51  5039.3  860.73  5090.5   864.1  5176.4  860.27  5220.2  860.69
  5735.9   864.3    5908  870.41  5970.5  873.03  6018.9  876.67  6126.6  882.81
  6225.3  881.72  6262.5  887.87  6333.2   889.9  6392.4  892.14  6428.7  893.44
#Mann= 16 ,-1 , 0
   601.5     .05       0   792.2     .05       0   911.3     .05       0
    2018     .05       0    3359     .05       0  4975.5     .05       0
  5025.5     .05       0  5039.3     .05       0  5176.4     .05       0
  5220.2     .05       0    5908     .05       0  5970.5     .05       0
  6018.9     .05       0  6225.3     .05       0  6333.2     .05       0
  6392.4     .05       0
#XS Ineff= 2 , 0
       0  2958.3  883.78               0
Permanent Ineff=
       F       F
Bank Sta=4975.5,5025.5
XS Rating Curve= 0 ,0
Exp/Cntr=0.3,0.1

Type RM Length L Ch R = 1 ,453375  ,1572,1572,1572
BEGIN DESCRIPTION:
Denton Creek 179.0
END DESCRIPTION:
XS GIS Cut Line= 3
      2244220.46      7212434.71      2240817.16      7211179.65
      2238343.33      7209226.77
#Sta/Elev= 30
  1001.1  919.73  1418.3  896.98  1450.3  890.44  2076.8  863.91  2446.1  855.42
  3826.7  856.61  4649.1  860.11  4690.3  860.02  4727.2  848.03  4840.9  856.31
  4882.7  856.73  4919.1  863.51  4946.8  860.75  4969.3  850.05  4971.5  844.71
  4975.5  843.71  5021.5  844.71  5025.4  853.06  5097.5  867.23  5147.2  860.09
  5238.5  858.27  5971.8  857.03  6399.2  859.15  6812.9  875.13  6883.4  883.31
  6983.1  880.04  7197.2  887.01  7202.4  887.06  7261.8  885.71  7780.2  931.38
#Mann= 10 ,-1 , 0
  1001.1     .05       0  2076.8     .05       0  3826.7     .05       0
  4649.1     .05       0  4840.9     .05       0  4971.5    .035       0
  5021.5     .05       0  5971.8     .05       0  7197.2     .16       0
  7202.4     .05       0
Bank Sta=4971.5,5021.5
XS Rating Curve= 0 ,0
Exp/Cntr=0.3,0.1

Type RM Length L Ch R = 1 ,451803  ,1399,1399,1399
BEGIN DESCRIPTION:
Denton Creek 178.0
END DESCRIPTION:
XS GIS Cut Line= 3
      2243379.03      7211360.03        2241379.        7209760.
        2239379.        7208360.
#Sta/Elev= 30
  2454.2  887.24  2539.9  882.62  2937.7  874.68  3072.9  869.04    3196  860.04
  3386.6  852.78    4349  857.96  4937.9  857.96  4944.3   857.7  4951.5  849.29
  4965.1   847.7  4968.9  841.07  4972.9  840.07  5018.9  841.07  5022.9  850.55
  5058.7  854.03    5145  856.06  5526.6  854.02  5656.3  854.45  5826.8  852.67
  6222.6  854.59  6315.1  857.64  6502.5  858.68  6675.1  864.87  6696.1   867.6
  6710.9  865.36  6782.4  864.81  7032.6  879.07  7398.8  912.05  7456.8  914.51
#Mann= 9 ,-1 , 0
  2454.2     .05       0  2937.7     .05       0    3196     .05       0
  3386.6     .05       0    4349     .05       0  4968.9    .035       0
  5018.9     .05       0  5526.6     .05       0  5656.3     .05       0
Bank Sta=4968.9,5018.9
XS Rating Curve= 0 ,0
Exp/Cntr=0.3,0.1

Type RM Length L Ch R = 1 ,450404  ,1418,1418,1418
BEGIN DESCRIPTION:
Denton Creek 177.0
END DESCRIPTION:
XS GIS Cut Line= 3
      2244428.98      7211009.98        2242429.        7209010.
       2240727.7      7207355.55
#Sta/Elev= 30
  2141.2   917.6  2452.3  898.44  2678.6   899.7  2862.4  884.44  3470.5  854.46
  3855.3  852.56  4657.3  852.49  4784.4  853.03    4913  856.87  4976.7  847.82
    4980  839.21    4984  838.21    5030  839.21  5033.3  850.01  5040.2  851.76
  5096.8  855.76  5683.8  853.29  5768.7  849.06  6050.3  868.38  6143.4   872.7
  6323.6  868.21  6412.2  872.97  6426.4  867.82  6454.7  870.76    6490  868.65
  6518.2  870.53  6532.4  876.78  6709.3  888.56  6992.2  896.85  7342.7   913.7
#Mann= 8 ,-1 , 0
  2141.2     .05       0  3855.3     .05       0  4657.3     .05       0
  4784.4     .05       0    4980     .05       0    5030     .05       0
  6050.3     .05       0  6323.6     .16       0
Bank Sta=4980,5030
XS Rating Curve= 0 ,0
Exp/Cntr=0.3,0.1

Type RM Length L Ch R = 1 ,448986  ,1394,1394,1394
BEGIN DESCRIPTION:
Denton Creek 176.0
END DESCRIPTION:
XS GIS Cut Line= 3
        2245083.      7209366.83        2243579.        7208210.
      2241578.99        7206610.
#Sta/Elev= 30
  3098.7  894.33  3199.2  883.19  3263.6  880.89  3298.9  883.35  3356.1   877.3
  3433.9   877.1  3620.6  866.32  3670.5  865.55  3712.1   869.7  3776.4  863.14
  3905.1  858.91  4482.3  849.25  4959.9  853.23    4968  834.24    4972  833.24
    5018  834.24  5025.2  847.23  5060.2  850.51  5102.6  848.14  5137.8  852.11
  5436.2  851.78  5597.8  851.64  6333.6  850.16    6352  847.49  6479.4  848.61
  6578.1   851.1    6789  866.19  7180.4  902.96  7455.1  911.36  7557.4  917.25
#Mann= 10 ,-1 , 0
  3098.7     .05       0    4968    .035       0    5018     .05       0
  5025.2     .05       0  5436.2     .05       0  5597.8     .05       0
    6352     .16       0  6479.4     .05       0  6578.1     .16       0
  7455.1     .05       0
Bank Sta=4968,5018
XS Rating Curve= 0 ,0
Exp/Cntr=0.3,0.1

Type RM Length L Ch R = 1 ,447592  ,1544,1544,1544
BEGIN DESCRIPTION:
Denton Creek 175.0
END DESCRIPTION:
XS GIS Cut Line= 3
      2245378.97      7208259.96        2244579.        7207260.
      2242281.77      7205063.68
#Sta/Elev= 30
  3737.6  880.67  3855.8  872.32  4091.7  855.26  4341.8  847.77  4961.4  852.09
  4967.8  850.17  4971.6  833.06  4975.6  832.06  5021.6  833.06  5025.3  837.12
  5039.4  843.22  5046.3   849.4  5055.3  851.01  5199.1  850.95  5349.1  850.57
  5463.7  847.99  5548.6  849.37    6300  846.07  6702.9  847.09  7267.4  846.76
  7451.4  856.07  7479.7  860.15  7550.1  862.91  7579.9  866.22  7649.2  873.75
  7769.6  881.38  7824.6   888.4  7946.2  899.67  8045.5  906.13  8196.4   898.5
#Mann= 13 ,-1 , 0
  3737.6     .05       0  3855.8     .05       0  4091.7     .05       0
  4971.6    .035       0  5021.6     .05       0  5055.3     .05       0
  5199.1     .05       0  5349.1     .05       0    6300     .05       0
  6702.9     .16       0  7579.9     .05       0  7824.6     .16       0
  7946.2     .05       0
Bank Sta=4971.6,5021.6
XS Rating Curve= 0 ,0
Exp/Cntr=0.3,0.1

Type RM Length L Ch R = 1 ,446048  ,2285,2285,2285
BEGIN DESCRIPTION:
Denton Creek 174.0
END DESCRIPTION:
XS GIS Cut Line= 3
      2246478.99      7208309.98      2245653.91       7205797.8
      2245078.99      7204709.98
#Sta/Elev= 30
  3022.7  884.41  3393.8  858.26    3570  859.65  3616.5  849.34  3637.3   849.3
  3748.7  848.41  3844.4  848.44  3959.4  857.27  3998.2  852.89  4235.4  850.99
  4267.9  850.29  4485.9  846.72  4902.4  848.52  4917.3  848.46  4931.3  837.87
  4948.8  847.06  4963.1  848.99  4976.5  833.74  4980.5  832.74  5026.5  833.74
  5026.7  841.51  5033.1  848.64  5090.4  851.59  5106.5   848.4  5368.4  850.05
  5433.8  849.97  6350.1  852.07  6467.5  848.84  6721.9  866.86  6897.3  884.15
#Mann= 12 ,-1 , 0
  3022.7     .05       0  3637.3     .05       0  3748.7     .05       0
  4235.4     .05       0  4267.9     .05       0  4902.4     .05       0
  4976.5    .035       0  5026.5     .05       0  5106.5     .16       0
  5368.4     .05       0  5433.8     .16       0  6721.9     .05       0
Bank Sta=4976.5,5026.5
XS Rating Curve= 0 ,0
Exp/Cntr=0.3,0.1

Type RM Length L Ch R = 1 ,443763  ,2001,2001,2001
BEGIN DESCRIPTION:
Denton Creek 172.0
END DESCRIPTION:
XS GIS Cut Line= 3
       2249295.7      7207720.42      2246620.34      7204850.34
      2245479.01        7204610.
#Sta/Elev= 30
    3053  891.38  3146.3  887.95  3376.5  876.73  3510.8  864.49  3567.5  863.56
    3631   869.5  3687.7  870.22  4013.1  852.62  4869.5  844.82  4918.8  850.14
  4940.2  846.32  4975.5  845.93  4978.9  827.24  4982.9  826.24  5028.9  827.24
  5032.2  832.13    5039  832.25  5053.2  838.51  5060.5  845.52    5103   847.4
  5279.9  844.83  5845.6  846.76  6769.7  854.23  7637.6  854.67  7685.1  853.73
  7744.5  856.46  7874.1  866.58  7973.8  870.21  8063.9  876.74    8143  874.02
#Mann= 7 ,-1 , 0
    3053     .05       0  3146.3     .05       0  4978.9     .05       0
  5028.9     .05       0  6769.7     .05       0  7637.6     .05       0
  8063.9     .05       0
Bank Sta=4978.9,5028.9
XS Rating Curve= 0 ,0
Exp/Cntr=0.3,0.1

Type RM Length L Ch R = 1 ,441762  ,1596,1596,1596
BEGIN DESCRIPTION:
Denton Creek 171.0
END DESCRIPTION:
XS GIS Cut Line= 3
      2251226.29      7206095.82      2249527.84      7205083.49
      2246301.15      7201544.37
#Sta/Elev= 30
  2704.9   882.8  3320.8   876.6  3325.8  876.47  3637.6   868.1  3896.5  848.53
  4799.5  840.32  4903.4  840.55  4924.5  833.59  4945.5   836.4  4952.9  830.49
  4959.7  834.91  4970.5  825.63  4974.5  824.63  5020.5  825.63  5030.6  841.05
  5044.8  843.27  5313.7  846.34  5802.2   848.9  5844.7  842.98  5901.5  848.29
  8367.7  852.52  8408.4  852.89    8598  854.63  8670.8  862.18    8931  873.31
  8994.6  867.53  9030.4  877.02  9259.2  892.72  9369.5  909.97  9471.4  914.95
#Mann= 11 ,-1 , 0
  2704.9     .05       0  3320.8     .05       0  3325.8     .05       0
  3637.6     .05       0  4799.5     .16       0  4970.5     .05       0
  5020.5     .16       0  8367.7     .05       0  8408.4     .05       0
  8670.8     .16       0  9259.2     .05       0
#XS Ineff= 2 , 0
       0                  6498.2       0   886.8
Permanent Ineff=
       F       F
Bank Sta=4970.5,5020.5
XS Rating Curve= 0 ,0
Exp/Cntr=0.3,0.1

Type RM Length L Ch R = 1 ,440166  ,308,308,308
BEGIN DESCRIPTION:
Denton Creek 170.0
END DESCRIPTION:
XS GIS Cut Line= 3
      2251635.75      7205102.01      2250704.38      7204034.11
      2248250.47      7201726.91
#Sta/Elev= 30
  2860.5  873.45  2980.4     866  3064.9  874.23  3136.1   863.2  3341.1  857.49
  3369.6  860.43  3412.4  855.44  3554.6  851.16  3901.3   843.4    4263  841.05
  4814.8  844.13  4878.3  851.64    4912  849.99  4970.6  844.02  4973.6  822.24
  4977.6  821.24  5023.6  822.24  5026.8  832.38  5055.2  844.09  5115.8  846.18
  6857.9  847.56  7007.8  853.24  7184.6  868.29  7283.8  865.99  7297.9  860.02
  7318.9  863.58  7340.4  858.86  7361.4  866.84  7503.1  877.52  7645.7  895.81
#Mann= 7 ,-1 , 0
  2860.5     .05       0  3554.6     .05       0    4912     .05       0
  4973.6    .035       0  5023.6     .05       0  5115.8     .05       0
  6857.9     .05       0
Bank Sta=4973.6,5023.6
XS Rating Curve= 0 ,0
Exp/Cntr=0.3,0.1

Type RM Length L Ch R = 1 ,439858  ,1825,1825,1825
BEGIN DESCRIPTION:
Denton Creek 169.0
END DESCRIPTION:
XS GIS Cut Line= 3
      2251847.24      7204833.81      2250759.94      7203660.57
      2248357.36      7201457.71
#Sta/Elev= 30
  2907.5   877.1  2916.3  876.95  2960.7  877.69  3021.9  870.79  3052.8  872.57
  3071.8  875.24  3156.8  873.86  3325.8   861.5  3530.1  848.34    3666  842.77
  4274.9  840.28  4914.7  846.52  4968.5  832.33  4971.8  820.37  4975.8  819.37
  5021.8  820.37  5024.6  844.43  5030.4  845.13  5060.3  845.53  5102.9  851.73
  5152.2  845.16  6617.3  845.75  6659.8  842.87  6928.7  871.07  6975.2  870.81
    7134  868.96  7346.1  885.98  7530.5  883.38  7650.7  898.75  7766.7  905.14
#Mann= 11 ,-1 , 0
  2907.5     .05       0  2916.3     .05       0  2960.7     .05       0
  3052.8     .05       0  3325.8     .05       0  3530.1     .05       0
  4914.7     .05       0  4971.8    .035       0  5021.8     .05       0
  5030.4     .05       0  6975.2     .05       0
Bank Sta=4971.8,5021.8
XS Rating Curve= 0 ,0
Exp/Cntr=0.3,0.1

Type RM Length L Ch R = 1 ,438033  ,1400,1400,1400
BEGIN DESCRIPTION:
Denton Creek 168.0
END DESCRIPTION:
XS GIS Cut Line= 3
      2253475.22      7202791.11        2251229.        7201760.
      2250508.82      7201310.35
#Sta/Elev= 30
  2513.1  869.28  2542.3  870.82  2650.1   875.6  2757.9  874.71  2865.7  870.18
  2948.1   866.2  2973.5  865.24  3081.3  861.41  3620.3  835.62  3794.5  839.32
  4099.9  841.53  4559.4     843  4841.6   842.5  4901.5  848.78  4940.7  842.58
  4952.9   836.7  4970.4  834.51  4973.2  818.25  4977.2  817.15  5023.2  818.25
  5028.9  836.48    5056  843.18  5223.5   840.5  5260.1  841.12  5340.9  847.45
  5442.9  856.44  5543.2  856.43  5714.3  861.73  5829.3  868.76  5833.7     869
#Mann= 15 ,-1 , 0
  2513.1     .05       0  2542.3     .05       0  2650.1     .05       0
  2757.9     .05       0  2865.7     .05       0  2948.1     .05       0
  2973.5     .05       0  3081.3     .05       0  4099.9     .05       0
  4559.4     .05       0  4973.2    .035       0  5023.2     .05       0
  5340.9     .05       0  5714.3     .05       0  5829.3     .05       0
Bank Sta=4973.2,5023.2
XS Rating Curve= 0 ,0
Exp/Cntr=0.3,0.1
