HEC-RAS study Harts Creek.prj: Harts Creek Base Level Engineering

--- Harts Creek.g01 (geometry) --- (continued)

Type RM Length L Ch R = 1 ,37849   ,395,395,395
BEGIN DESCRIPTION:
Harts Creek 64.0
END DESCRIPTION:
XS GIS Cut Line= 3
       2280728.1      7196077.51      2280283.52      7195847.73
      2279726.55      7196054.88
#Sta/Elev= 30
  4408.7  894.62  4531.5  889.57  4590.9  890.73  4730.3  890.14  4823.3  887.06
    4851  882.23  4895.3  880.77  4914.2  879.43    4930  876.68  4935.3  877.95
    4955  875.69  4960.3  876.31  4995.3  866.92    5010  868.25  5015.7  876.01
    5021  876.78  5031.3   885.6  5040.7  899.34    5046  897.24  5052.7   913.8
  5071.1  916.38  5076.4  915.52  5095.4   917.2  5198.9  918.13  5272.8  917.33
  5372.8  922.46  5413.9  923.23  5468.8  926.86  5478.2  928.58  5503.4  930.78
#Mann= 6 ,-1 , 0
  4408.7     .05       0  4730.3     .12       0    4955     .07       0
  5015.7     .12       0  5198.9     .12       0  5478.2     .05       0
Bank Sta=4960.3,5015.7
XS Rating Curve= 0 ,0
Exp/Cntr=0.3,0.1

Type RM Length L Ch R = 1 ,37454   ,509,509,509
BEGIN DESCRIPTION:
Harts Creek 63.0
END DESCRIPTION:
XS GIS Cut Line= 4
      2280736.23      7196056.79      2280518.37       7195760.3
      2280373.43      7195580.53      2280049.33      7195305.52
#Sta/Elev= 30
  4533.1  894.85  4686.5  886.85  4728.3  888.98  4839.8  887.36  4857.9  884.76
  4872.5  885.18  4878.7  883.06  4887.2   885.2  4893.4  884.78  4898.1  881.57
  4904.4  881.57  4907.9  878.46  4951.1  877.72  4957.5  877.12  4982.2  865.57
  5021.5  869.31  5035.9  878.03  5050.3  882.17  5071.1  884.06    5079  881.98
  5085.5  885.31  5120.7  889.77  5128.6  888.67  5185.3   891.3  5269.8  892.19
  5277.5  893.71  5284.1  891.77  5298.4   892.1  5354.2  895.38    5557  900.33
#Mann= 5 ,-1 , 0
  4533.1     .05       0  4839.8     .12       0  4951.1     .07       0
  5035.9     .12       0  5354.2     .05       0
Bank Sta=4957.5,5035.9
XS Rating Curve= 0 ,0
Exp/Cntr=0.3,0.1

Type RM Length L Ch R = 1 ,36945   ,404,404,404
BEGIN DESCRIPTION:
Harts Creek 62.0
END DESCRIPTION:
XS GIS Cut Line= 3
      2280872.24      7195509.17       2280614.4       7195293.7
      2280053.05       7195160.3
#Sta/Elev= 30
    4793  907.29  4801.6  907.99  4815.9  904.79  4830.2  899.05  4836.8  898.74
  4844.6  895.63  4879.7  892.02  4887.5  888.04    4894  888.55  4901.5  884.04
  4914.8  881.92  4922.6  883.76  4929.2  879.07    4937  880.25  4943.5  877.52
  4951.3  878.25  4957.8  875.33  4965.6  876.87  4972.1  870.34  4979.7  871.08
  4986.4   869.6  4996.7   862.8    5015  864.22  5029.4   873.7  5043.7  877.87
  5163.5  884.71  5239.5  885.53  5474.2  886.41  5642.9  890.29    5706  893.91
#Mann= 4 ,-1 , 0
    4793     .12       0  4965.6     .07       0  5043.7     .12       0
  5239.5     .05       0
Bank Sta=4965.6,5043.7
XS Rating Curve= 0 ,0
Exp/Cntr=0.3,0.1

Type RM Length L Ch R = 1 ,36541   ,473,473,473
BEGIN DESCRIPTION:
Harts Creek 61.0
END DESCRIPTION:
XS GIS Cut Line= 3
      2281176.35      7195003.08        2280729.        7195010.
      2280066.38      7195051.14
#Sta/Elev= 30
  4548.2  906.41  4615.6   903.5  4676.5  895.61  4715.6   893.7  4725.6   891.8
  4745.6  881.87  4755.6   886.4  4765.6  888.41  4795.6  888.49  4805.6  886.02
  4815.6  881.43  4825.6  880.63  4845.6  884.38  4875.6  881.14  4895.6  876.76
  4955.6  873.68  4998.1  866.31  5011.5  859.71  5019.7  859.71  5025.7  862.62
  5055.7  865.49  5073.5  869.99  5078.5  869.54  5095.8  872.57  5135.9  881.62
  5157.7   882.5  5306.2  881.39  5366.3  884.93  5516.6  887.46  5659.5   892.6
#Mann= 4 ,-1 , 0
  4548.2     .12       0  4955.6     .07       0  5095.8     .12       0
  5157.7     .05       0
Bank Sta=4955.6,5095.8
XS Rating Curve= 0 ,0
Exp/Cntr=0.3,0.1

Type RM Length L Ch R = 1 ,36068   ,346,346,346
BEGIN DESCRIPTION:
Harts Creek 60.0
END DESCRIPTION:
XS GIS Cut Line= 3
      2281072.24      7194662.67        2280579.        7194610.
      2280049.08      7194588.65
#Sta/Elev= 30
  4503.5  895.56  4521.9  895.39    4574  890.94  4587.2  890.85  4607.3  888.37
  4657.6   886.6  4687.8  883.34    4856  878.51  4929.1   874.2  4948.3  869.35
  4953.4  868.84  4959.3  863.63  4975.3  858.49  4983.5  858.49    4997  861.53
    5002  861.53  5029.6  868.74  5039.6  873.68  5049.6  878.23  5069.6  878.21
    5089  879.61  5149.7  881.44  5209.7   881.1  5289.8  883.89  5309.8  883.76
  5339.8  886.48  5359.8  886.33  5379.9  888.47  5439.9  891.49  5529.9   894.3
#Mann= 6 ,-1 , 0
  4503.5     .12       0  4521.9     .05       0    4856     .12       0
  4929.1     .07       0  5039.6     .12       0    5089     .05       0
Bank Sta=4929.1,5039.6
XS Rating Curve= 0 ,0
Exp/Cntr=0.3,0.1

Type RM Length L Ch R = 1 ,35722   ,516,516,516
BEGIN DESCRIPTION:
Harts Creek 59.0
END DESCRIPTION:
XS GIS Cut Line= 3
      2281110.64      7194444.86      2280624.46      7194327.44
      2279893.03      7194300.07
#Sta/Elev= 30
  4419.3  886.94  4513.6  881.12  4595.9  877.89  4678.8  877.04  4799.3  877.67
  4889.9  875.05  4924.9  874.33  4944.9  871.61    4965  865.09  4982.4  860.56
  5010.9  857.78  5020.6  858.28    5045  873.33    5055  876.06    5075  879.25
    5085  878.99  5105.1  880.16  5115.1   879.8  5138.2  881.45  5225.1  884.68
  5355.2  893.38  5375.2  893.97  5405.3  896.66    5520  901.03  5555.4  903.76
  5575.4   904.4  5595.4  905.95  5615.4  909.33  5635.4  908.93  5651.4  913.36
#Mann= 5 ,-1 , 0
  4419.3     .05       0  4889.9     .12       0  4924.9     .07       0
    5045     .12       0  5138.2     .05       0
Bank Sta=4924.9,5045
XS Rating Curve= 0 ,0
Exp/Cntr=0.3,0.1

Type RM Length L Ch R = 1 ,35206   ,441,441,441
BEGIN DESCRIPTION:
Harts Creek 58.0
END DESCRIPTION:
XS GIS Cut Line= 4
       2281148.6      7194429.67      2280825.47       7194201.4
      2280852.87      7193922.88      2280570.18      7193717.52
#Sta/Elev= 30
  4460.9  887.67  4488.7  886.37  4553.9  881.46  4696.7  874.89  4726.3  874.91
  4732.4  874.24  4741.1   874.7  4747.2     874    4762   873.9  4803.8  871.81
  4848.2  872.41  4942.8  870.37  4968.5  870.54  4978.5  866.48  4988.6   860.5
  4998.6  855.85  5004.5  854.63  5012.8  854.63  5018.7  857.06  5028.8  863.63
  5038.8  874.32  5044.8  875.63  5058.9  875.41    5069  876.24  5114.4  875.66
  5269.9     878    5406  882.76  5420.7  884.42  5441.5  884.91  5485.8  887.58
#Mann= 5 ,-1 , 0
  4460.9     .05       0  4942.8     .12       0  4968.5     .07       0
  5038.8     .12       0  5114.4     .05       0
Bank Sta=4968.5,5038.8
XS Rating Curve= 0 ,0
Exp/Cntr=0.3,0.1

Type RM Length L Ch R = 1 ,34765   ,456,456,456
BEGIN DESCRIPTION:
Harts Creek 57.0
END DESCRIPTION:
XS GIS Cut Line= 3
      2281287.07      7194226.66      2281077.68      7193805.59
      2280606.76      7193695.39
#Sta/Elev= 30
  4650.3  881.28  4668.9  879.46  4699.5  879.39    4705  878.14  4721.9  877.37
  4727.4  876.18  4811.5  870.98  4884.2  870.48    4901  868.44  4906.6   866.4
  4923.4  870.28  4936.9  868.97  4945.8   865.6  4951.4  865.72  4968.2  859.69
  4973.8  859.02  4981.6  855.54  4992.1   852.4  5000.4   852.4  5003.9  854.65
    5013  855.62  5018.6  857.87  5035.4  871.67    5041  874.06  5129.5  873.27
  5298.8  874.34  5431.4  878.38  5521.5  882.57    5564  883.02  5604.2  885.37
#Mann= 3 , 0 , 0
  4650.3     .05       0  4936.9    .033       0  5035.4     .05       0
Bank Sta=4936.9,5035.4
XS Rating Curve= 0 ,0
Exp/Cntr=0.3,0.1

Type RM Length L Ch R = 1 ,34309   ,497,497,497
BEGIN DESCRIPTION:
Harts Creek 56.0
END DESCRIPTION:
XS GIS Cut Line= 3
      2281667.53      7193636.46      2281332.05      7193636.65
      2280608.74      7193638.26
#Sta/Elev= 30
    4661  889.87  4689.5  886.28  4799.5  878.11  4809.5  876.62  4819.5  875.84
    4862  873.12  4909.5  869.44  4949.5  867.97  4959.5  866.42  4969.5  863.35
  4979.5  859.44  4989.5   854.3  4995.5   852.1  5000.5   852.1  5005.4  849.95
  5013.7  849.95  5015.3  850.45  5019.5  856.79  5029.5     863  5039.5  868.54
  5049.5   870.7  5069.5  869.48  5149.5  871.71  5259.5  872.45  5279.5  872.11
  5429.5  874.76  5549.5  878.68  5609.5  882.11  5639.5  882.43  5719.8  887.34
#Mann= 4 ,-1 , 0
    4661     .05       0    4862     .12       0  4949.5     .07       0
  5039.5     .05       0
Bank Sta=4949.5,5039.5
XS Rating Curve= 0 ,0
Exp/Cntr=0.3,0.1

Type RM Length L Ch R = 1 ,33812   ,406,406,406
BEGIN DESCRIPTION:
Harts Creek 55.0
END DESCRIPTION:
XS GIS Cut Line= 4
      2282034.98      7193345.69      2281593.41      7193197.65
      2281388.69      7193190.45      2280886.07      7193348.32
#Sta/Elev= 30
  4419.6  903.26    4458  899.33  4503.2  896.83  4599.2  889.72  4668.3  884.45
  4689.6  881.19  4705.1  880.42  4721.2  877.63  4752.9  874.43  4837.2  867.49
  4899.7  864.57  4955.2  864.44  4957.7  864.57  4962.7  864.25  4969.8  862.44
  4979.8  854.01    4984  848.47  4985.6  847.97  4993.9  847.97  5009.8  851.38
  5039.8  865.59  5048.6  866.73  5059.8  868.65  5330.9  868.56  5542.5  871.72
  5582.5  873.51  5602.1  877.61  5607.3  876.93  5612.8  880.61    5617  880.61
#Mann= 7 ,-1 , 0
  4419.6     .05       0  4503.2     .12       0  4599.2     .05       0
  4955.2     .12       0  4957.7     .07       0  5039.8     .12       0
  5048.6     .05       0
Bank Sta=4962.7,5039.8
XS Rating Curve= 0 ,0
Exp/Cntr=0.3,0.1

Type RM Length L Ch R = 1 ,33406   ,565,565,565
BEGIN DESCRIPTION:
Harts Creek 54.0
END DESCRIPTION:
XS GIS Cut Line= 3
      2281991.37       7192756.5        2281679.        7192910.
      2280878.98      7193310.01
#Sta/Elev= 30
  4648.1  878.89  4802.3  872.77  4852.8  872.15  4884.7  869.67  4892.2  870.76
  4920.3  870.26    4953  867.57  4987.7  863.81  4993.4   865.1  4998.9   865.1
  5004.5  862.75  5010.1  854.47  5018.5  850.91  5036.7  847.57  5046.6  848.07
  5071.6  855.96  5077.2  860.31  5116.3   864.9  5170.2   865.4  5256.1  867.03
  5577.5  868.01  5792.8  872.15  5837.5  873.99  5854.2  877.61  5859.8  877.21
  5868.2  879.71  5876.6  884.72  5882.2  883.77  5887.8  887.45  5890.6  887.45
#Mann= 5 ,-1 , 0
  4648.1     .05       0    4953     .12       0  4993.4     .07       0
  5116.3     .12       0  5170.2     .05       0
Bank Sta=4998.9,5116.3
XS Rating Curve= 0 ,0
Exp/Cntr=0.3,0.1

Type RM Length L Ch R = 1 ,32841   ,430,430,430
BEGIN DESCRIPTION:
Harts Creek 53.0
END DESCRIPTION:
XS GIS Cut Line= 3
      2281780.16      7192370.04      2281487.42       7192450.3
        2280729.        7192710.
#Sta/Elev= 30
  4602.5  868.13  4728.1  863.95  4877.8  862.15  4957.2  861.15    4983  859.82
  4988.9  858.95  4999.5  857.07    5009  852.14  5014.3  851.06    5027  845.26
  5035.4  845.26  5040.3  846.99  5045.6  846.99  5062.9  860.49  5071.6  863.93
  5084.1  864.55  5099.2  862.78  5126.3   862.1  5264.6  864.73  5384.4  869.32
  5478.3  874.08  5504.3  876.87    5528     877  5535.6   878.2  5603.5   880.8
  5634.8  886.52  5654.8  887.42  5686.6  890.98  5705.1  897.87  5707.7  897.87
#Mann= 5 ,-1 , 0
  4602.5     .05       0  4877.8     .12       0    4983     .07       0
  5071.6     .12       0  5099.2     .05       0
Bank Sta=4988.9,5071.6
XS Rating Curve= 0 ,0
Exp/Cntr=0.3,0.1

Type RM Length L Ch R = 1 ,32411   ,419,419,419
BEGIN DESCRIPTION:
Harts Creek 52.0
END DESCRIPTION:
XS GIS Cut Line= 4
      2281840.61       7192293.1      2281312.35      7192083.23
      2281230.87      7192265.83      2280922.49      7192368.82
#Sta/Elev= 30
  4352.2  872.17  4526.1  863.38  4673.6   861.8  4762.8  862.25  4917.3  857.35
    4928  858.49  4942.8  857.44    4966  857.78  4971.8  857.11  4982.8  846.09
  4989.2  844.02  5000.5  842.23  5008.9  842.23  5012.4  844.34  5035.7  847.95
  5041.1   847.4  5064.4  854.95  5081.3  857.78  5275.6  864.97  5344.1  866.43
    5365  868.14  5370.4   869.8  5375.7   868.9  5386.1  870.95    5402  872.49
  5407.3  872.08  5428.3  876.96  5433.6  879.99  5438.9  879.59  5445.7  882.22
#Mann= 4 ,-1 , 0
  4352.2     .05       0  4673.6     .12       0    4966     .07       0
  5081.3     .05       0
Bank Sta=4966,5081.3
XS Rating Curve= 0 ,0
Exp/Cntr=0.3,0.1

Type RM Length L Ch R = 1 ,31992   ,449,449,449
BEGIN DESCRIPTION:
Harts Creek 51.0
END DESCRIPTION:
XS GIS Cut Line= 4
      2281848.32      7192280.98      2281273.83      7192011.86
      2281250.66      7191855.79      2281057.42      7191594.57
#Sta/Elev= 30
  4211.5  872.84  4386.3  863.54  4528.4  862.28  4694.1  858.82  4716.9  856.27
  4722.4  853.24  4739.7  855.92  4745.3  852.19  4762.6  857.39  4768.1  851.97
  4773.9  855.57    4785  857.03  4913.2  857.27  4938.8  855.65    4959  851.91
  5019.1   840.7  5045.2  842.93  5066.1  851.44  5080.7  851.03  5086.9  853.46
  5095.3  849.25  5101.6  854.03    5110  850.77  5116.2  852.33  5122.8  851.06
    5137  857.66  5145.4  865.02  5160.1  870.32  5266.5  872.35  5328.6  876.13
#Mann= 4 ,-1 , 0
  4211.5     .05       0  4528.4     .12       0    4959     .07       0
  5066.1     .12       0
Bank Sta=4959,5066.1
XS Rating Curve= 0 ,0
Exp/Cntr=0.3,0.1

Type RM Length L Ch R = 1 ,31543   ,427,427,427
BEGIN DESCRIPTION:
Harts Creek 50.0
END DESCRIPTION:
XS GIS Cut Line= 3
      2281892.63      7192190.16      2281478.64      7191861.48
       2281049.6      7191485.15
#Sta/Elev= 30
  4475.2   875.1  4569.8  870.27  4577.8  868.91  4598.6  869.01  4620.3  865.91
  4662.7  863.74  4670.7  864.27  4697.9  861.83    4748  861.95    4762  860.67
  4791.5  860.71  4811.8  860.37  4834.1  861.95  4840.5  860.06  4862.9  859.77
  4898.2   854.5  4926.7  845.53  4954.3  841.56  4964.5  837.66  4974.5  838.16
  4976.7  841.46  4983.1  844.65  4990.6  850.46    5001  855.54  5060.5  860.12
  5089.6  862.27  5146.6   864.2  5408.5   869.4  5514.8  875.78  5574.5   884.8
#Mann= 5 ,-1 , 0
  4475.2     .05       0  4791.5     .12       0  4898.2     .07       0
    5001     .12       0  5060.5     .05       0
Bank Sta=4898.2,5001
XS Rating Curve= 0 ,0
Exp/Cntr=0.3,0.1

Type RM Length L Ch R = 1 ,31116   ,296,296,296
BEGIN DESCRIPTION:
Harts Creek 49.0
END DESCRIPTION:
XS GIS Cut Line= 3
      2282034.33      7191525.21        2281629.        7191510.
      2281103.78      7191452.25
#Sta/Elev= 30
  4594.4  867.62  4619.8  865.06  4709.8  860.34  4799.9  857.81  4848.9  857.96
  4899.9  858.08    4940  855.51    4950  854.08    4960  850.99    4970  848.83
    4980  845.67    4990  840.76  4993.3  840.03  5001.8  840.03  5020.1     845
  5040.3  847.24  5045.5  851.34  5050.6  854.37  5060.4  857.28  5080.5  854.56
  5175.2  858.01  5191.2  859.09  5241.5  859.53  5301.8  861.71  5402.4  867.54
  5409.6   868.5  5462.8     872    5493  874.62  5513.1  878.83  5528.4  881.25
#Mann= 5 ,-1 , 0
  4594.4     .05       0  4848.9     .12       0    4940     .07       0
  5060.4     .12       0  5175.2     .05       0
Bank Sta=4940,5060.4
XS Rating Curve= 0 ,0
Exp/Cntr=0.3,0.1

Type RM Length L Ch R = 1 ,30820   ,244,244,244
BEGIN DESCRIPTION:
Harts Creek 48.1
END DESCRIPTION:
XS GIS Cut Line= 2
      2282060.18      7191236.42      2281216.43      7191192.26
#Sta/Elev= 30
  4568.3  863.31  4619.5  859.23  4649.6  857.84  4749.7  855.69  4803.2  856.21
  4839.8  855.96  4849.9  856.44    4920  855.53    4950  852.94    4960  852.96
    4970  850.02    4975   847.1  4981.6  845.62  4990.1  839.26  5005.8  836.03
  5014.3  836.03  5015.9  836.53  5020.1  842.84  5040.1  851.71  5060.2  851.81
  5158.3  854.94  5190.3  855.53  5200.3  854.94  5260.4  858.02  5280.5   858.2
  5291.7  859.17  5330.5   861.4  5350.5  863.23  5363.2  863.01  5413.2  866.66
#Mann= 6 ,-1 , 0
  4568.3     .05       0  4803.2     .12       0    4960     .07       0
  5040.1     .12       0  5158.3     .05       0  5291.7     .12       0
Bank Sta=4960,5040.1
XS Rating Curve= 0 ,0
Exp/Cntr=0.3,0.1

Type RM Length L Ch R = 1 ,30576   ,378,378,378
BEGIN DESCRIPTION:
Harts Creek 48.0
END DESCRIPTION:
XS GIS Cut Line= 4
      2282130.08      7191133.65      2281771.42      7191011.49
      2281498.68      7190975.36      2281058.16      7190745.71
#Sta/Elev= 30
    4427   867.7  4618.3  854.52  4717.6  854.67  4927.9  853.31  4932.9  853.13
  4985.7  835.64  4994.2  835.64  5006.3  839.94  5011.4  838.43  5050.4  848.46
  5078.3  851.36    5081  851.36    5084  849.48  5144.7   854.1  5213.4  855.32
  5245.3  856.38  5315.8   858.7  5328.8  851.77  5337.9     850  5343.5  852.99
  5365.6  856.81  5382.1  850.17  5396.4  855.71  5404.2  861.48  5409.8  862.37
  5492.5  864.64  5520.5  860.59  5536.7   861.8  5565.6  870.89  5577.8  871.66
#Mann= 6 ,-1 , 0
    4427     .05       0  4717.6     .12       0  4927.9     .07       0
    5081     .12       0  5213.4     .05       0  5245.3     .12       0
Bank Sta=4932.9,5078.3
XS Rating Curve= 0 ,0
Exp/Cntr=0.3,0.1

Type RM Length L Ch R = 1 ,30198   ,425,425,425
BEGIN DESCRIPTION:
Harts Creek 47.0
END DESCRIPTION:
XS GIS Cut Line= 3
      2282028.15      7191072.06        2281679.        7190710.
      2281306.86      7190408.71
#Sta/Elev= 30
  4502.3     859  4609.2  853.85    4680  852.47  4686.9  851.59    4749  852.18
  4764.9  851.63  4771.8  852.81    4786  853.02  4793.2   852.1  4856.7  852.66
  4934.7  847.39  4941.6  848.11  4948.8  843.97  4955.8  841.84  4972.9  833.76
  4981.4  833.76  4998.2  836.72  5001.8   841.2  5008.5   841.2  5018.9  849.84
  5026.9  850.86  5088.6  852.53  5211.2   856.6  5247.5  856.27  5282.7  858.14
  5354.9  858.91  5410.6  859.73  5439.3  861.51  5460.1  861.27  5484.1  862.48
#Mann= 6 ,-1 , 0
  4502.3     .05       0    4749     .12       0  4934.7     .07       0
  5018.9     .12       0  5088.6     .05       0  5354.9     .12       0
Bank Sta=4941.6,5018.9
XS Rating Curve= 0 ,0
Exp/Cntr=0.3,0.1

Type RM Length L Ch R = 1 ,29773   ,496,496,496
BEGIN DESCRIPTION:
Harts Creek 46.0
END DESCRIPTION:
XS GIS Cut Line= 3
      2282207.66      7190389.83        2281829.        7190360.
      2281279.04        7190360.
#Sta/Elev= 30
  4624.6  873.84  4633.3  872.53  4703.5  866.92  4816.2  858.71  4843.9  855.51
  4894.1   852.4  4914.3  846.62  4924.2  845.31  4934.2  843.16    4940  839.05
  4980.1  834.72  4988.6  834.72  4990.3  835.22  4994.4  838.63  5001.9  842.38
  5006.9  842.38  5014.4  849.52  5084.4  847.63  5154.4  846.95  5214.4  848.16
  5244.4  849.36  5304.4  854.23  5344.4  854.41  5374.4  855.73  5384.4  854.97
  5464.4  859.04  5534.4  864.51  5544.4  866.05  5551.9  868.92  5554.4  868.92
#Mann= 4 ,-1 , 0
  4624.6     .05       0  4914.3     .12       0  4924.2     .07       0
  5014.4     .12       0
Bank Sta=4924.2,5014.4
XS Rating Curve= 0 ,0
Exp/Cntr=0.3,0.1

Type RM Length L Ch R = 1 ,29277   ,408,408,408
BEGIN DESCRIPTION:
Harts Creek 45.0
END DESCRIPTION:
XS GIS Cut Line= 3
      2282132.16       7190087.8      2281796.99      7190051.62
      2281207.74      7190002.58
#Sta/Elev= 30
  4594.6  879.55  4616.8  881.05    4628  880.58    4638  879.33  4648.1  875.94
  4698.4  865.35  4718.7   862.2  4748.6  860.84  4768.8  857.29  4829.1   851.5
  4871.5  849.26  4939.7  847.12  4949.8  844.99  4969.8   837.6    4974  830.39
  4975.6  829.89  4984.2  829.89  4999.9  832.63  5013.3  838.35    5030  843.51
  5154.4  849.14  5170.5  850.42  5230.7  851.76  5331.1  857.52  5391.3  861.58
  5431.4   865.5  5471.6  867.71  5490.2   870.1  5501.7   868.8    5523  869.96
#Mann= 5 ,-1 , 0
  4594.6     .05       0  4871.5     .12       0  4939.7     .07       0
    5030     .12       0  5154.4     .05       0
Bank Sta=4939.7,5030
XS Rating Curve= 0 ,0
Exp/Cntr=0.3,0.1

Type RM Length L Ch R = 1 ,28869   ,250,250,250
BEGIN DESCRIPTION:
Harts Creek 44.0
END DESCRIPTION:
XS GIS Cut Line= 3
      2282128.99      7189859.99        2281829.        7189710.
      2281369.56       7189491.6
#Sta/Elev= 30
  4660.3  879.29  4668.7  877.89  4674.3  878.54    4691  871.99    4705  868.72
  4713.4  864.81    4719  865.26  4727.4  860.36  4735.8  858.82  4780.5  853.15
  4852.7  846.71  4892.3  840.78  4897.9  844.22  4914.6  842.35  4920.2  844.44
  4942.6   841.7    4951  838.42  4973.3  835.27  4987.3  830.53    5000  828.94
  5010.2  829.44  5017.8  837.27    5027  843.06  5049.7  844.13  5055.3  841.75
  5062.1  843.99  5086.7  845.91    5129  846.29  5327.9  853.46  5504.4  864.49
#Mann= 5 ,-1 , 0
  4660.3     .05       0  4852.7     .12       0  4942.6     .07       0
    5027     .12       0  5086.7     .05       0
Bank Sta=4942.6,5027
XS Rating Curve= 0 ,0
Exp/Cntr=0.3,0.1

Type RM Length L Ch R = 1 ,28619   ,285,285,285
BEGIN DESCRIPTION:
Harts Creek 43.0
END DESCRIPTION:
XS GIS Cut Line= 3
      2282215.47      7189742.32      2281908.57      7189484.76
      2281463.13      7189145.64
#Sta/Elev= 30
  4595.6  869.04  4858.6  846.04  4943.1  841.37  4991.8  828.33    5028  830.12
  5034.3  836.35  5042.5  832.08  5063.4  835.12  5077.9  842.69  5098.7  835.49
  5113.3  839.95  5134.1  835.72  5156.9   842.4  5163.2  837.74  5171.4  841.43
  5177.7  838.13  5192.2  849.73  5227.6  844.76  5242.1  852.71  5271.2  854.34
  5277.5  850.34    5292  855.52    5371  856.57  5377.3  852.84  5391.8  858.78
  5448.2  850.63  5470.8   855.4  5520.7  854.66  5541.5  863.13  5556.1   856.1
#Mann= 4 ,-1 , 0
  4595.6     .05       0  4858.6     .12       0  4943.1     .07       0
  5034.3     .12       0
Bank Sta=4943.1,5034.3
XS Rating Curve= 0 ,0
Exp/Cntr=0.3,0.1

Type RM Length L Ch R = 1 ,28334   ,314,314,314
BEGIN DESCRIPTION:
Harts Creek 42.1
END DESCRIPTION:
XS GIS Cut Line= 2
      2282367.45      7189465.75       2281522.8      7188951.85
#Sta/Elev= 30
  4612.6  865.39  4615.3  864.49    4658  860.64  4673.5  860.35  4739.5   853.2
  4783.9  850.73  4805.2  848.06  4857.8  844.63    4906  842.96  4921.4  844.36
  4927.3  842.96  4942.7  842.52  4958.2  836.35  4964.1  835.36  4975.2  827.82
  4983.8  827.82  5000.9  829.99  5008.8  831.91  5022.2  836.98  5043.9  842.16
  5125.8  844.75  5132.6  846.37  5148.1   846.1  5190.7  848.58  5242.9  849.78
  5328.3  853.46  5386.4  857.03  5488.7     861    5587  867.93  5601.3  869.86
#Mann= 5 ,-1 , 0
  4612.6     .05       0  4857.8     .12       0  4942.7     .07       0
  5043.9     .12       0    5587     .05       0
Bank Sta=4942.7,5043.9
XS Rating Curve= 0 ,0
Exp/Cntr=0.3,0.1

Type RM Length L Ch R = 1 ,28020   ,237,237,237
BEGIN DESCRIPTION:
Harts Creek 42.0
END DESCRIPTION:
XS GIS Cut Line= 3
      2282579.04      7189260.02        2282129.        7189010.
      2281629.02      7188710.01
#Sta/Elev= 30
  4489.3  883.36  4535.1  876.13  4562.6  867.67  4578.6  859.22  4584.3  859.48
  4600.3  852.73  4615.2  850.63    4622  851.91  4630.1  850.63  4659.8  851.09
    4725  845.33  4790.2  842.48  4855.4  841.57  4930.9  843.47  4946.9  839.78
  4958.4  831.91  4976.9  827.41  4987.2  827.91  4996.1  839.52  5001.3  843.66
  5120.7  841.89  5229.6  845.12  5272.4  848.08  5287.9  847.64  5478.4  860.91
  5493.9  862.88  5515.3  868.72  5521.1  867.95  5562.4  871.31  5587.2  873.24
#Mann= 5 ,-1 , 0
  4489.3     .05       0  4630.1     .12       0  4930.9     .07       0
  5001.3     .12       0  5562.4     .05       0
Bank Sta=4930.9,5001.3
XS Rating Curve= 0 ,0
Exp/Cntr=0.3,0.1

Type RM Length L Ch R = 1 ,27783   ,497,497,497
BEGIN DESCRIPTION:
Harts Creek 41.2
END DESCRIPTION:
XS GIS Cut Line= 3
      2282651.75      7189224.01      2282154.19      7188710.07
      2281557.82      7188496.46
#Sta/Elev= 30
  4443.7  886.96  4462.7  885.16  4476.9  881.95  4483.8   878.1    4498  873.94
  4526.3   869.7  4533.2  865.14  4547.4  861.39  4576.3  856.51  4653.6  847.74
  4717.2  843.01  4943.5  840.25  4957.7  837.34  4964.6  833.44  4995.8  827.17
  5006.1  827.67  5007.1  837.62  5014.3  836.62  5021.2  841.61  5028.4  842.72
  5233.5  839.59  5419.5  846.33  5493.8  851.71  5530.5  857.18  5568.2  866.39
  5598.4  869.43  5673.7  870.33    5679   869.3  5704.4  871.83  5792.5  875.67
#Mann= 5 ,-1 , 0
  4443.7     .05       0  4576.3     .12       0  4943.5     .07       0
  5028.4     .12       0  5598.4     .05       0
Bank Sta=4943.5,5021.2
XS Rating Curve= 0 ,0
Exp/Cntr=0.3,0.1

Type RM Length L Ch R = 1 ,27286   ,602,602,602
BEGIN DESCRIPTION:
Harts Creek 41.1
END DESCRIPTION:
XS GIS Cut Line= 3
      2283253.62      7188039.17      2282273.68      7188460.38
      2281655.85      7188510.61
#Sta/Elev= 30
  3737.1  842.81  3959.9  838.68  4211.6  838.76  4253.3  837.37  4701.6   839.9
  4715.2  840.68  4767.8  839.09  4838.5   840.4  4848.6  841.77  4898.7   840.5
  4908.8  841.81  4948.9  841.52  4958.9  840.46    4969  838.19  4984.1  830.88
  5013.3   825.3    5025   825.3  5049.2   831.6  5069.3  838.91  5089.3  841.76
  5209.7  851.07  5259.9  853.19    5280  858.14    5300  860.34  5320.1   865.9
  5322.8  865.52  5330.1  864.51  5360.2  868.05  5390.3  866.97  5423.6   869.6
#Mann= 5 ,-1 , 0
  3737.1     .05       0  4701.6     .12       0  4948.9     .07       0
  5089.3     .12       0  5322.8     .05       0
Bank Sta=4958.9,5089.3
XS Rating Curve= 0 ,0
Exp/Cntr=0.3,0.1

Type RM Length L Ch R = 1 ,26684   ,433,433,433
BEGIN DESCRIPTION:
Harts Creek 41.0
END DESCRIPTION:
XS GIS Cut Line= 5
      2283332.41      7188012.38      2282486.94      7188009.29
        2282329.        7188060.       2282165.9      7188084.07
      2281782.29      7188049.29
#Sta/Elev= 30
  3984.7  845.47  4368.1  837.42  4468.1  837.86  4558.1  836.53  4678.1  837.46
  4883.7   835.8  4922.5  837.51  4951.9  837.18    4980  839.24  4985.6  838.12
  4993.4  829.84  4998.6  829.84  5006.2  823.56  5010.4  821.86  5025.8  822.47
  5036.5  826.15  5056.7   829.2  5066.8  832.18  5100.5  833.67  5107.2  837.25
  5137.6  837.59  5187.9  842.85  5218.1  842.69  5248.2  845.25  5278.5   845.6
  5338.5  848.94  5372.9  849.36  5428.9  854.07    5459  852.67  5546.1  859.18
#Mann= 5 ,-1 , 0
  3984.7     .05       0  4951.9     .12       0  4985.6     .07       0
  5107.2     .12       0  5278.5     .05       0
#XS Ineff= 2 , 0
       0    4980  839.24  5117.4       0  837.99
Permanent Ineff=
       F       F
Bank Sta=4985.6,5107.2
XS Rating Curve= 0 ,0
Exp/Cntr=0.3,0.1

Type RM Length L Ch R = 1 ,26251   ,442,442,442
BEGIN DESCRIPTION:
Harts Creek 40.0
END DESCRIPTION:
XS GIS Cut Line= 5
      2283386.97      7187927.21       2282537.9      7187849.62
        2282379.        7187710.      2282260.62      7187608.81
      2281744.42      7187655.72
#Sta/Elev= 30
  3935.6  848.04  4325.2  837.67  4385.4  837.77  4465.8  835.68    4526  837.52
  4566.2   835.8  4636.5   836.2  4656.6  837.66  4686.7   836.1  4777.1   837.1
  4794.3   836.1  4815.2   838.4  4861.5  836.45    4929  835.22  4978.4  827.87
    5003  826.06  5015.2  820.72    5029  821.22  5035.4  828.28  5049.7  834.39
    5064  837.74  5228.1  837.22  5307.7  841.82  5333.6  844.57  5449.1  846.83
  5528.6  851.05  5559.6  854.63  5574.8  854.42    5629  855.24  5673.8  857.86
#Mann= 5 ,-1 , 0
  3935.6     .05       0  4861.5     .12       0    4929     .07       0
  5049.7     .05       0  5574.8     .12       0
Bank Sta=4929,5049.7
XS Rating Curve= 0 ,0
Exp/Cntr=0.3,0.1

Type RM Length L Ch R = 1 ,25809   ,453,453,453
BEGIN DESCRIPTION:
Harts Creek 39.0
END DESCRIPTION:
XS GIS Cut Line= 3
      2283433.08      7187295.64        2282579.        7187460.
      2281807.19      7187556.75
#Sta/Elev= 30
  4134.2   866.7  4168.9  861.55    4184  856.12  4189.3  851.32    4230     850
    4241  850.98  4270.7  846.09  4362.4  840.32  4566.1   835.7  4596.6  836.69
  4667.9  834.56  4739.2  834.59  4759.5   832.9  4872.7  834.29    4921  836.12
  4926.1  836.19    4953  826.19  4963.2  825.32  4964.9  820.59  4966.9  820.09
  4978.8  820.09  5001.4  828.96  5040.6   834.2  5074.5  835.44  5165.2  833.95
  5306.3  836.45  5467.6  837.09  5524.7  841.56  5669.1  847.66  5781.8  854.33
#Mann= 5 ,-1 , 0
  4134.2     .05       0  4872.7     .12       0    4921     .07       0
  5040.6     .12       0  5040.6     .05       0
Bank Sta=4926.1,5040.6
XS Rating Curve= 0 ,0
Exp/Cntr=0.3,0.1

Type RM Length L Ch R = 1 ,25356   ,447,447,447
BEGIN DESCRIPTION:
Harts Creek 38.0
END DESCRIPTION:
XS GIS Cut Line= 4
      2283353.45      7187045.72        2282729.        7187060.
      2282370.36      7187082.84      2281962.49      7187270.37
#Sta/Elev= 30
  4375.3  855.76  4419.8  850.72  4459.8  850.13  4489.8  844.87  4539.8  838.84
  4569.8  839.26  4629.8  835.79    4783  831.65  4799.9  829.72  4839.9  832.08
  4887.8  832.87  4929.9  835.87  4939.9  834.68  4959.9  828.52    4974  819.17
  4985.9  819.17  5002.4  821.58  5009.9  824.21    5030  835.02  5035.6  836.04
    5040  836.85  5070.1  833.88  5150.2  832.34  5220.4  833.55  5290.5  830.94
  5503.2  832.22    5669  836.19    5721  839.43  5772.5  840.58  5808.2  844.65
#Mann= 5 ,-1 , 0
  4375.3     .05       0  4887.8     .12       0  4929.9     .07       0
    5030     .12       0  5035.6     .05       0
Bank Sta=4929.9,5030
XS Rating Curve= 0 ,0
Exp/Cntr=0.3,0.1

Type RM Length L Ch R = 1 ,24909   ,315,315,315
BEGIN DESCRIPTION:
Harts Creek 37.0
END DESCRIPTION:
XS GIS Cut Line= 4
      2283347.62      7186755.79      2282717.08      7186609.34
      2282617.35      7186782.66      2281916.27      7187060.15
#Sta/Elev= 30
  4286.1  852.11  4448.9  838.91  4582.4  834.67  4651.7  834.95  4731.4  830.92
  4767.2  832.49  4774.1  831.89  4779.2  827.76  4787.7  832.17  4816.7  827.34
  4821.8  829.37  4921.2   833.9  4945.7  832.85  4958.8  828.87  4961.3  828.71
  4968.8  824.65  4976.7  816.72  4991.1  817.22  4991.9  819.45  4998.7  823.26
  5004.5  820.22  5072.6   829.4  5107.3   827.9  5116.5  828.71  5122.3  832.07
  5138.4   832.7  5400.5  826.13  5516.8  826.14  5768.1  835.88  5887.4  846.23
#Mann= 4 ,-1 , 0
  4286.1     .05       0  4651.7     .12       0  4958.8     .05       0
  5072.6     .05       0
Bank Sta=4961.3,5072.6
XS Rating Curve= 0 ,0
Exp/Cntr=0.3,0.1

Type RM Length L Ch R = 1 ,24594   ,67,67,67
BEGIN DESCRIPTION:
Harts Creek 36.3
END DESCRIPTION:
XS GIS Cut Line= 6
      2283354.75      7186692.22      2282490.25       7186518.8
      2282428.23       7186510.4      2282336.25      7186557.56
      2282031.11      7186563.66       2281632.9      7186839.52
#Sta/Elev= 30
  4057.4   847.8  4091.4  845.34  4096.5  843.38  4142.3  842.88  4147.4  840.03
  4193.3   840.7    4346  835.38    4453  835.73  4517.7   833.8    4563  831.17
  4695.6  835.23  4718.9  833.81  4906.2  829.84    4920  831.42  4966.5   825.6
  4971.6  828.62  4980.8  826.06  4992.6  817.75  5031.3  821.41  5053.5  828.01
  5090.7  831.57  5105.1  829.98  5132.3   832.4  5230.7  829.01  5312.9  828.69
  5473.7  833.89  5546.7   840.9  5631.8  842.34  5854.3  854.71  5894.7  855.24
#Mann= 7 ,-1 , 0
  4057.4     .05       0  4517.7     .12       0  4718.9     .05       0
  4966.5    .033       0  5053.5     .05       0  5230.7     .12       0
  5312.9     .05       0
Bank Sta=4971.6,5053.5
XS Rating Curve= 0 ,0
Exp/Cntr=0.3,0.1

Type RM Length L Ch R = 1 ,24527   ,446,446,446
BEGIN DESCRIPTION:
Harts Creek 36.2
END DESCRIPTION:
XS GIS Cut Line= 6
      2283314.12      7186611.29      2282458.34      7186439.27
      2282407.01      7186451.76      2282319.32      7186505.44
      2282227.72      7186513.64      2281643.79      7186524.81
#Sta/Elev= 30
  4044.9  846.95  4128.1  842.49  4498.6  833.33  4850.2  830.83  4892.3  832.43
  4897.5  830.81  4937.4   830.4  4942.5  832.02  4948.1  832.34  4991.2  825.56
  5003.3  821.14  5015.7  820.03  5017.9   816.2  5019.9   815.7  5034.3   816.2
  5040.3  826.16  5049.3  827.54  5055.3  831.98  5071.2  831.96    5084  833.05
    5104  827.46  5114.1  826.63  5188.3  826.34  5233.1   825.2  5604.4  841.46
  5664.4  840.54  5684.4  838.01  5704.4  832.97  5734.4   848.1  5749.6  848.54
#Mann= 5 ,-1 , 0
  4044.9     .05       0  4942.5    .033       0  5055.3     .05       0
  5071.2     .12       0  5188.3     .05       0
Bank Sta=4948.1,5055.3
XS Rating Curve= 0 ,0
Exp/Cntr=0.3,0.1

Type RM Length L Ch R = 1 ,24081   ,505,505,505
BEGIN DESCRIPTION:
Harts Creek 36.1
END DESCRIPTION:
XS GIS Cut Line= 3
      2283145.68      7186456.67       2282399.5      7186109.11
      2281628.18      7186324.94
#Sta/Elev= 30
  3794.1   840.5    3978  832.87  4512.8  828.57  4562.6  826.98  4614.8  828.71
  4700.8  826.73  4763.1  827.75  4783.1  825.85  4794.3  822.23  4901.1  826.36
  4974.6  824.19  4981.2   823.9    5002  821.24  5008.7  817.91  5026.9  814.14
  5053.9  816.38  5074.7  827.16  5082.1  830.36  5087.3  826.51  5105.8  833.65
  5155.6  833.18  5220.1  837.07  5234.2  836.42  5251.2  827.56  5261.6  827.69
  5273.6  832.82  5292.7  836.35  5386.4  844.87    5407  848.39  5418.2  847.89
#Mann= 4 ,-1 , 0
  3794.1     .05       0  4512.8     .12       0  4974.6     .07       0
  5082.1     .05       0
#XS Ineff= 2 , 0
       0                  5220.1       0  837.07
Permanent Ineff=
       F       F
Bank Sta=4981.2,5074.7
XS Rating Curve= 0 ,0
Exp/Cntr=0.3,0.1

Type RM Length L Ch R = 1 ,23576   ,440,440,440
BEGIN DESCRIPTION:
Harts Creek 36.0
END DESCRIPTION:
XS GIS Cut Line= 3
      2283144.37      7186370.95        2282279.        7185960.
      2281606.73      7185841.63
#Sta/Elev= 30
  4038.3  839.04  4119.2  835.08  4221.4  832.32  4803.2  827.51  4896.8  827.01
    4965  828.22  4974.1  823.99  4982.2  816.24  4985.2  812.11  4987.2  811.61
  4999.8  811.61  5023.4  818.07  5057.2   822.9    5108  823.23  5136.9  821.83
  5158.8  822.64  5189.2  821.89  5219.7  823.16  5295.5  822.91  5314.8  824.18
  5321.2  827.44  5331.4   830.4  5351.7  831.68  5412.6  832.65  5473.5   835.9
  5487.6  835.52  5541.8   837.6  5554.8  836.81  5625.8  842.18  5678.9  842.13
#Mann= 5 ,-1 , 0
  4038.3     .05       0  4803.2     .12       0    4965     .07       0
  5057.2     .12       0  5295.5     .05       0
Bank Sta=4974.1,5057.2
XS Rating Curve= 0 ,0
Exp/Cntr=0.3,0.1

Type RM Length L Ch R = 1 ,23136   ,112,112,112
BEGIN DESCRIPTION:
Harts Creek 35.0
END DESCRIPTION:
XS GIS Cut Line= 4
      2283395.78      7186433.58      2282135.76      7185558.75
      2282005.62      7185683.02      2281597.62      7185811.05
#Sta/Elev= 30
  3389.9  849.84  3404.6  847.67  3476.2  846.03  3526.8  842.77  3547.8   843.3
  3562.6  841.17  3613.3  839.16  3857.8  832.48  4021.9  830.32  4194.8  829.63
  4266.4  830.84  4331.9  828.34    4469   826.7  4741.2   826.2  4862.7   826.1
  4907.3  827.62  4923.8  826.19  4929.6  825.97  4950.7  822.23  4957.9  817.82
  4979.9  811.32  4992.5  811.32  5014.5  815.31  5028.7   819.9  5049.7  821.43
  5085.3  827.07  5106.6  826.97  5307.7  830.94  5512.7  841.48  5531.4  844.96
#Mann= 5 ,-1 , 0
  3389.9     .05       0  4741.2     .12       0  4923.8     .07       0
  5085.3     .12       0  5106.6     .05       0
#XS Ineff= 2 , 0
       0  4266.4  830.84               0
Permanent Ineff=
       F       F
Bank Sta=4929.6,5085.3
XS Rating Curve= 0 ,0
Exp/Cntr=0.3,0.1

Type RM Length L Ch R = 1 ,23024   ,213,213,213
BEGIN DESCRIPTION:
Harts Creek 34.3
END DESCRIPTION:
XS GIS Cut Line= 4
      2282927.98      7185274.41      2282214.82      7185329.76
      2281951.98      7185577.84      2281566.67      7185763.66
#Sta/Elev= 30
  3990.4   840.2    4210  830.74  4330.4  826.91  4470.8  825.45  4670.2  826.99
  4745.3  827.72  4752.6  825.55  4766.7  818.94  4780.9  818.07  4801.9  826.42
  4809.2  827.82  4858.6  824.87  4922.1  825.91  4929.4  825.24  4936.2   821.3
  4943.5  814.24  4950.4  814.99  4958.2  811.83  4970.8  811.83  4978.7  816.38
    4986  816.89  5000.2  815.09  5021.2  819.16  5042.6  819.54  5065.7  824.98
    5108  827.34  5131.3  827.33  5214.8  828.65  5339.6  832.92  5494.9  844.83
#Mann= 5 ,-1 , 0
  3990.4     .05       0  4670.2     .12       0  4922.1     .07       0
  5065.7     .12       0  5131.3     .05       0
#XS Ineff= 2 , 0
       0  4809.2  827.82               0
Permanent Ineff=
       F       F
Bank Sta=4929.4,5065.7
XS Rating Curve= 0 ,0
Exp/Cntr=0.3,0.1

Type RM Length L Ch R = 1 ,22811   ,72,72,72
BEGIN DESCRIPTION:
Harts Creek 34.2
END DESCRIPTION:
XS GIS Cut Line= 3
       2282937.9      7185205.31      2282084.33      7185228.92
      2281488.85      7185655.49
#Sta/Elev= 30
  3841.8  841.55  3950.7  835.03  3990.8  834.11  4170.8  826.74  4230.8  826.09
  4330.9  826.78  4400.9   824.8    4531  825.81  4589.4  825.21    4681  825.77
  4742.9   819.9  4772.4  824.68  4914.9  824.96  4923.4  824.49  4959.1  817.48
  4986.1  810.88  4986.3   809.8  4988.3   809.3    5003   809.8  5009.4  811.53
  5015.6  815.11  5030.3  820.17  5051.2  825.28  5068.1  825.69  5116.3  826.11
  5122.4  827.09    5131  826.76  5158.1   828.5  5258.8  831.82  5428.2  846.09
#Mann= 5 ,-1 , 0
  3841.8     .05       0  4589.4     .12       0  4914.9     .07       0
  5051.2     .12       0  5068.1     .05       0
#XS Ineff= 2 , 0
       0  4800.7  824.87               0
Permanent Ineff=
       F       F
Bank Sta=4923.4,5051.2
XS Rating Curve= 0 ,0
Exp/Cntr=0.3,0.1

Type RM Length L Ch R = 1 ,22739   ,285,285,285
BEGIN DESCRIPTION:
Harts Creek 34.1
END DESCRIPTION:
XS GIS Cut Line= 3
      2282938.26      7185171.55      2282027.18        7185186.
      2281332.75      7185682.23
#Sta/Elev= 30
  3821.5  842.59  3990.8  832.18  4076.9   829.2  4114.4  827.65  4310.8  826.63
  4370.8  824.42  4594.1  826.07  4742.4  825.17  4763.3  823.14  4769.4  819.16
  4784.2   817.9  4813.7  818.67  4834.5  823.48  4855.4  824.65  4950.1  823.84
  4977.1  816.49  5006.6  815.29  5029.7  808.69  5044.4  809.19    5050  815.41
    5057  819.58  5071.7  823.82  5079.2  824.67  5300.3  833.83  5329.8  836.07
  5335.9  838.35  5466.2  848.25  5493.2  852.99  5552.2  855.44  5586.2  859.62
#Mann= 6 ,-1 , 0
  3821.5     .05       0  4076.9     .12       0  4114.4     .05       0
  4594.1     .12       0  4950.1     .07       0  5079.2     .05       0
#XS Ineff= 2 , 0
       0    4864  824.77               0
Permanent Ineff=
       F       F
Bank Sta=4950.1,5071.7
XS Rating Curve= 0 ,0
Exp/Cntr=0.3,0.1

Type RM Length L Ch R = 1 ,22454   ,243,243,243
BEGIN DESCRIPTION:
Harts Creek 34.0
END DESCRIPTION:
XS GIS Cut Line= 3
      2282975.69      7185130.79      2281782.09      7185067.16
      2281304.43      7185187.16
#Sta/Elev= 30
  3803.1  844.66  3913.4  839.74  4040.1  830.42  4083.1  829.23  4130.3  826.86
    4193  826.28  4230.4  826.07  4240.4  827.91  4270.5  825.85  4320.5  826.09
  4360.6  824.36  4531.7  825.14  4630.9  824.78  4863.3  822.41  4931.4  820.33
  4941.4  818.85  4961.4  810.98  4965.1  808.09  4991.5  810.24  4997.4  813.58
  5002.6  813.58  5022.2  823.46    5029  825.51  5041.5  825.23  5166.6  827.71
  5234.1   831.2    5281  832.54    5337  837.92  5445.5  842.42  5490.9  846.47
#Mann= 11 ,-1 , 0
  3803.1     .05       0  4083.1     .12       0    4193     .05       0
  4531.7     .12       0  4630.9     .05       0  4863.3     .12       0
  4931.4     .07       0  5022.2     .12       0  5041.5     .05       0
  5234.1     .12       0    5337     .05       0
#XS Ineff= 2 , 0
       0  4240.4  827.91               0
Permanent Ineff=
       F       F
Bank Sta=4931.4,5022.2
XS Rating Curve= 0 ,0
Exp/Cntr=0.3,0.1

Type RM Length L Ch R = 1 ,22211   ,442,442,442
BEGIN DESCRIPTION:
Harts Creek 33.0
END DESCRIPTION:
XS GIS Cut Line= 3
      2283079.02        7185060.        2281879.        7184860.
      2281509.03       7184763.2
#Sta/Elev= 30
  3779.2  852.67  3819.8  850.54  3867.9  845.75    3911   845.6  3994.7  841.35
  4141.7   830.9  4265.8  821.57  4316.5  825.24  4419.1   824.4  4448.3  826.04
  4542.1  823.81  4785.4   823.6  4895.1  819.93  4934.9  821.31  4962.8   819.6
  4967.9  819.41  4993.2  811.34  4998.4  811.34    5007  807.32  5021.9  807.82
  5047.5  820.79  5053.8  820.78    5059  823.17  5094.3  825.96  5154.4  827.32
  5175.1  829.48  5210.4  830.24  5305.9  841.34  5331.7     841  5378.2  844.34
#Mann= 7 ,-1 , 0
  3779.2     .05       0  4141.7     .12       0  4419.1     .05       0
  4895.1     .12       0  4962.8     .07       0  5047.5     .12       0
  5154.4     .05       0
#XS Ineff= 2 , 0
       0  4448.3  826.04               0
Permanent Ineff=
       F       F
Bank Sta=4967.9,5047.5
XS Rating Curve= 0 ,0
Exp/Cntr=0.3,0.1

Type RM Length L Ch R = 1 ,21769   ,454,454,454
BEGIN DESCRIPTION:
Harts Creek 32.0
END DESCRIPTION:
XS GIS Cut Line= 3
      2283067.09      7184695.33        2282079.        7184510.
      2281878.98      7184459.99
#Sta/Elev= 30
    3995  852.07  4155.1   843.8  4212.8  839.06  4247.4  839.55  4267.1  836.02
    4323  832.79    4400  825.85  4428.1  819.81  4433.2  821.52  4450.9  817.94
  4485.8  815.49  4501.8  818.12    4512  821.89  4538.2  822.21  4847.7  822.81
  4949.5  819.48  4973.5   808.2  4986.4   808.2  4990.1  810.56  4997.8  811.89
  5023.5   813.2  5059.6  819.87  5082.8  822.63  5113.7   829.3  5127.7  829.92
  5147.2  829.78  5175.6  833.22  5183.3  836.13  5188.4   835.3  5206.5  837.37
#Mann= 6 ,-1 , 0
    3995     .05       0  4267.1     .12       0  4538.2     .05       0
  4949.5     .07       0  5059.6     .12       0  5127.7     .05       0
Bank Sta=4949.5,5059.6
XS Rating Curve= 0 ,0
Exp/Cntr=0.3,0.1

Type RM Length L Ch R = 1 ,21315   ,450,450,450
BEGIN DESCRIPTION:
Harts Creek 31.0
END DESCRIPTION:
XS GIS Cut Line= 3
      2282964.64      7184178.32        2282229.        7184110.
      2281903.02      7184088.33
#Sta/Elev= 30
  4261.6  834.62  4367.7  826.27  4404.2  824.97  4458.1  817.91  4468.1  815.12
  4478.2  813.26  4508.3  812.99  4538.4  819.34  4602.4  820.38  4628.8  821.12
  4658.9  820.57  4699.1  821.38  4799.5  820.66  4889.9  820.99  4940.1  820.17
  4960.2  821.01  4980.3  814.21  4989.4  805.87  4991.4  805.37  5004.3  805.37
  5030.5  812.85  5050.5   816.6  5060.5  819.33  5080.7  819.98  5096.5  822.29
  5120.7  825.95  5180.8  832.46  5220.9  832.83  5226.2  833.74  5327.1  838.33
#Mann= 5 ,-1 , 0
  4261.6     .12       0  4602.4     .05       0  4960.2     .07       0
  5060.5     .12       0  5096.5     .05       0
Bank Sta=4960.2,5060.5
XS Rating Curve= 0 ,0
Exp/Cntr=0.3,0.1

Type RM Length L Ch R = 1 ,20865   ,450,450,450
BEGIN DESCRIPTION:
Harts Creek 30.0
END DESCRIPTION:
XS GIS Cut Line= 3
      2283035.36      7183787.68        2282229.        7183660.
      2281917.82      7183662.45
#Sta/Elev= 30
  4183.6   827.7  4332.7  823.87    4459  818.82  4493.8  818.59  4524.8  816.61
  4534.3  815.09  4544.4  811.77  4554.5  809.81  4574.8  809.85  4605.1  815.06
  4615.3  816.87  4625.4  816.71  4649.5  810.17  4655.8  811.52  4665.9  815.44
  4696.3  818.08  4898.5  819.17  4959.5  820.95  4966.3  815.84  4971.4  816.02
    4989  804.66    4991  804.16  5005.9  804.66    5010   808.7    5020  813.33
    5030  817.87    5040  820.39  5109.4   822.4    5190  828.09  5311.2  832.68
#Mann= 7 ,-1 , 0
  4183.6     .05       0    4459     .12       0  4605.1     .05       0
  4898.5     .12       0  4959.5     .07       0    5040     .12       0
  5109.4     .05       0
Bank Sta=4959.5,5040
XS Rating Curve= 0 ,0
Exp/Cntr=0.3,0.1

Type RM Length L Ch R = 1 ,20415   ,531,531,531
BEGIN DESCRIPTION:
Harts Creek 29.0
END DESCRIPTION:
XS GIS Cut Line= 3
      2283439.65      7183445.33        2282229.        7183210.
      2281734.05        7183245.
#Sta/Elev= 30
  3766.8  845.42  4080.6  826.34  4132.2  825.41  4137.3  823.91  4292.4  815.78
  4439.8  813.58  4460.2  809.62  4480.6  810.32  4511.1   806.2  4531.5  808.63
  4550.7  815.38  4575.8  816.26  4755.6  815.44  4865.8   818.1  4954.9  815.53
  4969.2  814.63  4974.3  814.58  4991.1  803.26  5006.1  803.76  5020.2  813.13
  5030.2  816.68  5050.2  817.33  5090.3  813.84  5200.6  816.97  5231.4  819.85
  5260.8  822.32  5290.8  821.92  5300.9  823.66  5421.2  831.17  5496.3  834.25
#Mann= 6 ,-1 , 0
  3766.8     .12       0  4575.8     .05       0  4954.9     .12       0
  4969.2     .07       0  5030.2     .12       0  5231.4     .05       0
Bank Sta=4974.3,5030.2
XS Rating Curve= 0 ,0
Exp/Cntr=0.3,0.1

Type RM Length L Ch R = 1 ,19884   ,567,567,567
BEGIN DESCRIPTION:
Harts Creek 28.0
END DESCRIPTION:
XS GIS Cut Line= 4
      2283678.98      7183409.99      2282341.87      7182793.89
        2282129.        7182760.      2281728.99        7182710.
#Sta/Elev= 30
  3311.9  904.56  3320.6  901.07  3326.1  904.71  3343.6  894.96  3349.1   897.4
  3355.9  889.29  3366.5  885.53    3372  886.93    3395  871.52  3417.9  863.06
  3486.8  851.76  3532.1  847.33  3801.8  830.52    3945  818.51  4088.3  812.03
  4111.3  809.14  4225.7  814.15  4323.4  813.26  4351.9  810.75  4387.2  814.77
  4909.8  814.33    4949  814.29  4979.4  807.71  4990.6   802.2  5005.6   802.7
  5019.8  811.44  5029.9  813.23    5119  816.51  5198.7  825.15  5402.8  834.42
#Mann= 6 ,-1 , 0
  3311.9     .12       0  4387.2     .05       0  4909.8     .12       0
    4949     .07       0  5029.9     .12       0    5119     .05       0
Bank Sta=4949,5029.9
XS Rating Curve= 0 ,0
Exp/Cntr=0.3,0.1

Type RM Length L Ch R = 1 ,19317   ,565,565,565
BEGIN DESCRIPTION:
Harts Creek 27.0
END DESCRIPTION:
XS GIS Cut Line= 3
      2283329.01      7183110.01        2282529.        7182510.
      2281729.01        7182010.
#Sta/Elev= 30
    4000  836.14  4021.9  831.59  4036.5  830.43  4057.3  830.48  4107.3  825.53
  4292.7  814.94  4363.6  809.12    4400  808.09  4436.5  812.39  4471.9  813.53
  4592.7  813.27  4678.1   809.2  4707.3  812.39    4714   811.4  4894.9  812.82
  4936.5  813.98  4942.7  813.88    4950  811.63  4965.4  801.91  4978.4  801.91
  4986.5  805.28  4996.9  807.05  5007.7  806.64  5013.6  813.32    5385  813.01
  5496.7  815.32  5530.7  815.87  5640.4  825.38  5731.7  829.31  5943.4  842.94
#Mann= 7 ,-1 , 0
    4000     .12       0    4714     .05       0  4894.9     .12       0
  4936.5    .033       0  5013.6     .12       0  5496.7     .12       0
  5640.4     .05       0
Bank Sta=4942.7,5013.6
XS Rating Curve= 0 ,0
Exp/Cntr=0.3,0.1

Type RM Length L Ch R = 1 ,18752   ,567,567,567
BEGIN DESCRIPTION:
Harts Creek 26.0
END DESCRIPTION:
XS GIS Cut Line= 4
        2283779.        7183060.        2282979.        7182260.
      2282819.29      7182112.86      2281745.84      7181932.66
#Sta/Elev= 30
  3868.9   907.3    3883  906.63  3897.2  901.18  3911.3  891.25  3928.1  882.79
  3939.6  875.07  3967.9  867.51  4024.5   857.4  4203.1  844.59  4307.3  840.09
  4335.6  836.08  4386.3   833.8  4519.4  824.88  4533.6  822.45    4576  820.28
  4604.3  821.93  4618.4  818.11  4717.4  813.37  4943.7  809.68  4965.4  798.99
  4980.5  799.49  4996.7  809.03  5000.3  809.03  5030.4  811.95  5155.9  808.83
  5717.5  812.63  5730.9  812.99  5817.6  814.67  6036.1  827.39  6305.9  844.01
#Mann= 11 ,-1 , 0
  3868.9     .05       0  3928.1     .12       0  4203.1     .05       0
  4386.3     .12       0  4943.7     .07       0  5000.3     .12       0
  5030.4     .05       0  5717.5     .12       0  5730.9     .05       0
  5817.6     .12       0  6036.1     .05       0
Bank Sta=4943.7,4996.7
XS Rating Curve= 0 ,0
Exp/Cntr=0.3,0.1

Type RM Length L Ch R = 1 ,18185   ,553,553,553
BEGIN DESCRIPTION:
Harts Creek 25.0
END DESCRIPTION:
XS GIS Cut Line= 3
      2283827.14      7181869.95        2283079.        7181760.
      2281629.02        7181660.
#Sta/Elev= 30
  4243.9  852.73  4277.7  849.54  4691.2  823.19  4787.8  815.99  4848.5  812.64
  4931.3   810.4  4939.4  810.65  4949.5  808.08  4965.2  800.74  4970.2  801.45
  4971.3  799.23  4973.3  798.73  4986.5  798.73  5030.1  808.71  5160.5  807.42
  5364.7  809.83  5471.2     809  5721.8   812.6  5872.1  817.05  5932.3  820.48
  6012.5  827.14  6072.6  829.38  6088.9  831.72  6142.8  834.27  6162.8  837.27
  6236.8  840.58    6243  842.29  6283.1  843.09  6303.2  846.17  6453.5  855.39
#Mann= 4 ,-1 , 0
  4243.9     .05       0  4931.3     .12       0  4949.5    .033       0
  5030.1     .05       0
Bank Sta=4949.5,5030.1
XS Rating Curve= 0 ,0
Exp/Cntr=0.3,0.1

Type RM Length L Ch R = 1 ,17632   ,583,583,583
BEGIN DESCRIPTION:
Harts Creek 24.0
END DESCRIPTION:
XS GIS Cut Line= 3
      2283849.06      7181339.44        2283229.        7181260.
      2282213.74      7181206.53
#Sta/Elev= 30
  4370.7  857.35  4639.8  834.88  4663.1   833.9  4693.4  830.46  4713.5  833.33
  4719.5  832.13  4724.5  829.07  4753.9  827.97  4887.5  817.49  4958.5  812.64
  4975.7  808.18  4985.7  804.54  4993.3  799.89  4995.8  799.89  4997.2  797.81
  4999.2  797.31  5012.4  797.31  5015.9  799.44  5035.9  805.87  5055.9   808.5
    5116  806.08  5196.1  807.25  5376.4   805.2  5446.5  806.43  5706.8  806.89
  5736.9  808.38  5846.7  819.22  5977.2   822.2  5997.2  826.58  6012.5  827.06
#Mann= 4 ,-1 , 0
  4370.7     .05       0  4887.5     .12       0  4975.7    .033       0
  5055.9     .05       0
Bank Sta=4975.7,5055.9
XS Rating Curve= 0 ,0
Exp/Cntr=0.3,0.1

Type RM Length L Ch R = 1 ,17049   ,525,525,525
BEGIN DESCRIPTION:
Harts Creek 23.0
END DESCRIPTION:
XS GIS Cut Line= 3
      2283804.15      7180588.35        2283129.        7180710.
      2282116.18      7180909.47
#Sta/Elev= 30
  4318.2  846.12  4333.6  841.92  4352.3  839.18  4410.9  833.28  4445.4  832.76
  4464.5  829.53  4469.6  830.78    4486  827.76  4523.2   824.5  4557.1  823.68
  4668.9  815.72  4694.2  815.31  4719.7  812.65  4752.9  812.68  4806.5  807.28
  4878.9  805.51  4963.6  806.73  4972.3  801.86  4995.1  798.22  5010.3  798.72
  5014.4  802.59  5024.6     807  5086.3  805.28  5381.3  804.35  5599.9  805.83
  5778.8  810.22  5805.3  813.17  5880.7  817.47    5908  820.66  6036.5   826.6
#Mann= 4 ,-1 , 0
  4318.2     .05       0  4878.9     .12       0  4963.6    .035       0
  5024.6     .05       0
Bank Sta=4963.6,5024.6
XS Rating Curve= 0 ,0
Exp/Cntr=0.3,0.1
