--- Miller Creek.prj (project) ---

Proj Title=Miller Creek Base Level Engineering
Current Plan=p01
Default Exp/Contr=0.3,0.1
English Units
Geom File=g01
Flow File=f01
Plan File=p01
Y Axis Title=Elevation
X Axis Title(PF)=Main Channel Distance
X Axis Title(XS)=Station
BEGIN DESCRIPTION:
Miller Creek
END DESCRIPTION:
DSS File=dss
DSS Export Rating Curves= 0
DSS Export Rating Curve Sorted= 0
DSS Export Volume Flow Curves= 0
DXF OffsetX= 0
DXF OffsetY= 0
DXF ScaleX= 1
DXF ScaleY= 10

--- Miller Creek.p01 (plan) ---

Plan Title=Multiple Run
Program Version=4.10
Short Identifier=Multiple Run
Geom File=g01
Flow File=f01
Subcritical Flow
K Sum by GR= 0
Std Step Tol= 0.01
Critical Tol= 0.01
Num of Std Step Trials= 20
Max Error Tol= 0.3
Flow Tol Ratio= 0.001
Split Flow NTrial= 30
Split Flow Tol= 0.02
Split Flow Ratio= 0.02
Log Output Level= 0
Friction Slope Method= 1
Unsteady Friction Slope Method= 2
Unsteady Bridges Friction Slope Method= 1
Parabolic Critical Depth
Global Vel Dist= 1 , 1 , 1
Global Log Level= 0
CheckData=True
Encroach Param=-1 ,0,0, 0
BEGIN DESCRIPTION:
Multiple Run
END DESCRIPTION:
Computation Interval=1HOUR
Output Interval=1HOUR
Run HTab= 0
Run UNet= 0
Run PostProcess= 0
Run WQNet= 0
UNET Theta= 1
UNET Theta Warmup= 1
UNET ZTol= 0.02
UNET ZSATol= 0.05
UNET MxIter= 20
UNET MaxInSteps= 0
UNET DtIC= 0
UNET DtMin= 0
UNET MaxCRTS= 20
UNET WFStab= 2
UNET SFStab= 1
UNET WFX= 1
UNET SFX= 1
UNET DSS MLevel= 4
UNET DZMax Abort= 100
UNET Convert EG Bridges= 0
UNET Use Existing IB Tables=-1
UNET Froude Reduction=False
UNET Froude Limit= 1
UNET Froude Power= 10
UNET Time Slicing=0,0, 5
UNET Junction Losses=0
Instantaneous Interval=1HOUR
DSS File=dss
Write IC File= 0
Write IC File at Sim End=0
Echo Input=False
Echo Parameters=False
Echo Output=False
Write Detailed= 0
WQ AD Non Conservative
WQ ULTIMATE=-1
WQ Max Comp Step=1HOUR
WQ Output Interval=15MIN
WQ Output Selected Increments= 0
WQ Output face flow=0
WQ Output face velocity=0
WQ Output face area=0
WQ Output face dispersion=0
WQ Output cell volume=0
WQ Output cell surface area=0
WQ Output cell continuity=0
WQ Output cumulative cell continuity=0
WQ Output face conc=0
WQ Output face dconc_dx=0
WQ Output face courant=0
WQ Output face peclet=0
WQ Output face adv mass=0
WQ Output face disp mass=0
WQ Output cell mass=0
WQ Output cell source sink temp=0
WQ Output cell source sink nsm=0
WQ Output MaxMinRange=-1
WQ Daily Max Min Mean=-1
WQ Daily Range=0
WQ Daily Time=0
WQ Create Restart=0
WQ Fixed Restart=0
WQ System Summary=0
WQ Use Fixed Temperature=0
Sorting and Armoring Iterations= 10
XS Update Threshold= 0.02
Hydraulics Update Threshold= 0.02
Energy Slope Method= 1
Volume Change Method= 0
XS Weighting Method= 0
Number of US Weighted Cross Sections= 1
Number of DS Weighted Cross Sections= 1
Upstream XS Weight=0.25
Main XS Weight=0.5
Downstream XS Weight=0.25
Number of DS XS's Weighted with US Boundary= 1
Upstream Boundary Weight= 1
Weight of XSs Associated with US Boundary= 0
Number of US XS's Weighted with DS Boundary= 1
Downstream Boundary Weight= 0.5
Weight of XSs Associated with DS Boundary= 0.5
Sediment Output Level= 4
Mass or Volume Output= 0
Output Increment Type= 1
Profile and TS Output Increment= 10
XS Output Flag= 0
XS Output Increment= 10
Disregard all LS=0
Disregard all Conn=0
Disregard all Breaches=0
Disregard all Pumps=0

--- Miller Creek.f01 (steady flow) ---

Flow Title=Multiple
Program Version=4.10
Number of Profiles= 7
Profile Names=10-year,25-year,50-year,1pct_min,100-year,1pct_plu,500-year
River Rch & RM=Miller Creek,Reach-1         ,18494
     628     865    1061     647    1291    2576    1914
River Rch & RM=Miller Creek,Reach-1         ,13498
     933    1311    1631    1007    2009    4009    3056
River Rch & RM=Miller Creek,Reach-1         ,6842
    1516    2184    2763    1731    3453    6891    5412
River Rch & RM=Miller Creek,Reach-1         ,4860
    1703    2467    3130    1967    3925    7831    6188
River Rch & RM=Miller Creek,Reach-1         ,4126
    1785    2590    3291    2071    4132    8244    6531
Boundary for River Rch & Prof#=Miller Creek,Reach-1         , 1
Up Type= 0
Dn Type= 3
Dn Slope=0.005
Boundary for River Rch & Prof#=Miller Creek,Reach-1         , 2
Up Type= 0
Dn Type= 3
Dn Slope=0.005
Boundary for River Rch & Prof#=Miller Creek,Reach-1         , 3
Up Type= 0
Dn Type= 3
Dn Slope=0.005
Boundary for River Rch & Prof#=Miller Creek,Reach-1         , 4
Up Type= 0
Dn Type= 3
Dn Slope=0.005
Boundary for River Rch & Prof#=Miller Creek,Reach-1         , 5
Up Type= 0
Dn Type= 3
Dn Slope=0.005
Boundary for River Rch & Prof#=Miller Creek,Reach-1         , 6
Up Type= 0
Dn Type= 3
Dn Slope=0.005
Boundary for River Rch & Prof#=Miller Creek,Reach-1         , 7
Up Type= 0
Dn Type= 3
Dn Slope=0.005
DSS Import GetInterval= 0
DSS Import GetPeak= 0
DSS Import FillOption= 0

--- Miller Creek.g01 (geometry) ---

Geom Title=Existing Conditions
Program Version=4.10

River Reach=Miller Creek    ,Reach-1
Reach XY= 30
        2288129.        7201010.      2287532.67      7199758.41
      2287424.01        7199108.      2287130.05      7199048.38
      2287228.75      7198775.22      2286980.26      7198350.29
      2287078.68      7197925.02      2286875.49      7197211.25
      2286530.99      7197104.73      2286971.92      7195959.98
      2286432.31      7195701.98      2286329.47      7195273.71
      2286525.48      7195011.46      2285889.19      7194719.68
      2286021.51      7194456.42      2285586.62       7194116.5
      2285573.59      7193815.17       2285186.8      7193816.21
      2285278.29      7193469.79      2285078.52      7193230.16
        2285229.        7193010.      2284722.46       7193051.1
      2284709.87      7192539.58        2284079.        7192360.
      2283975.85       7191467.7      2283181.09      7190304.74
      2283223.64       7189557.3      2282882.66      7189351.83
      2282802.34      7188883.05        2282279.        7188660.

Type RM Length L Ch R = 1 ,18494   ,100,100,100
BEGIN DESCRIPTION:
Miller Creek 44.0
END DESCRIPTION:
XS GIS Cut Line= 2
      2288359.63      7200773.78      2287772.96       7201179.7
#Sta/Elev= 30
  4700.4  991.22  4704.9  989.43  4713.3  989.67  4719.8  988.75  4725.8  989.42
  4749.5  988.12  4791.4  988.06  4806.3  986.44  4812.3     987  4821.1  985.71
  4827.2  985.95  4842.1  984.73  4956.5   980.3  4970.5  978.26  4985.3  977.88
    4991  974.58  4991.3  974.08    4995  974.58  5000.2   977.2  5006.3  977.44
  5042.1  978.44  5078.1  978.34  5143.5  980.18  5158.3  981.88    5209  984.44
  5215.1  986.37  5223.9  985.75  5244.8  985.92  5337.4  989.49  5413.8  991.32
#Mann= 3 ,-1 , 0
  4700.4     .05       0    4991    .033       0    4995     .05       0
Bank Sta=4991,4995
XS Rating Curve= 0 ,0
Exp/Cntr=0.3,0.1

Type RM Length L Ch R = 1 ,18394   ,294,294,294
BEGIN DESCRIPTION:
Miller Creek 43.0
END DESCRIPTION:
XS GIS Cut Line= 2
      2288368.38      7200701.55      2287671.27      7201075.55
#Sta/Elev= 30
  4671.6   989.3  4677.7  988.61  4683.4   989.1  4699.7  987.16  4705.3  987.86
  4721.6  987.43  4737.8  986.03  4750.3  986.63  4759.8  985.06  4765.4   985.7
  4803.6  983.52  4809.3  984.43  4825.5  982.88  4831.2  983.52  4935.2  979.55
  4957.1  977.63  4973.3  975.13    4979  975.49  4995.3  973.77  4998.9  972.74
  4999.2  972.24  5002.7  972.24  5002.9  972.74  5011.3  974.94  5022.9  975.68
  5055.4  975.82  5136.2  977.86  5186.9  981.96  5283.7  986.44  5462.7   989.7
#Mann= 3 ,-1 , 0
  4671.6     .05       0  4998.9    .033       0  5002.9     .05       0
Bank Sta=4998.9,5002.9
XS Rating Curve= 0 ,0
Exp/Cntr=0.3,0.1

Type RM Length L Ch R = 1 ,18100   ,300,300,300
BEGIN DESCRIPTION:
Miller Creek 42.0
END DESCRIPTION:
XS GIS Cut Line= 2
      2288253.58      7200366.98      2287669.39      7200860.41
#Sta/Elev= 30
  4632.7     991  4645.2  991.25  4673.8  989.03  4694.6   988.4  4751.8  985.28
  4772.6  985.05  4780.4  984.27  4801.2  983.82  4829.8  981.68  4850.6  981.04
  4872.7  979.67  4893.5  977.81  4900.5  976.74  4907.8  976.49  4928.7  973.74
    4965  972.73    4977  970.94  4977.3  970.44  4980.8  970.44    4981  970.94
  5000.1  972.19    5043  972.34  5084.7  973.99  5092.4  974.84  5106.7  975.42
  5135.3  975.47    5177  977.79  5248.5  980.36    5333   984.3  5397.4  985.33
#Mann= 3 ,-1 , 0
  4632.7     .05       0    4977    .033       0    4981     .05       0
Bank Sta=4977,4981
XS Rating Curve= 0 ,0
Exp/Cntr=0.3,0.1

Type RM Length L Ch R = 1 ,17800   ,255,255,255
BEGIN DESCRIPTION:
Miller Creek 41.0
END DESCRIPTION:
XS GIS Cut Line= 2
      2288292.29      7200323.75      2287199.44       7200358.2
#Sta/Elev= 30
  4586.5  993.75  4599.8  993.51  4649.8  989.67  4679.8  987.81  4689.8  987.59
  4729.9  984.62  4819.9  977.24  4859.9  973.34    4900  971.37    4910  971.36
    4930   969.6    4980  969.57    5000  969.93    5090   969.6  5120.1  970.28
  5140.1  969.44  5238.1   969.4  5238.4   968.9  5241.9   968.9  5242.1   969.4
  5340.2  969.54  5360.2  972.83  5370.2  973.91  5390.2  975.33  5430.2     979
  5450.2  979.56  5470.2  981.17  5576.8  984.63  5581.8  984.47  5679.9  989.23
#Mann= 3 ,-1 , 0
  4586.5     .05       0  5238.1    .033       0  5242.1     .05       0
Bank Sta=5238.1,5242.1
XS Rating Curve= 0 ,0
Exp/Cntr=0.3,0.1

Type RM Length L Ch R = 1 ,17545   ,131,131,131
BEGIN DESCRIPTION:
Miller Creek 40.0
END DESCRIPTION:
XS GIS Cut Line= 3
      2288014.94      7200141.53        2287729.        7200160.
      2287442.46      7200186.53
#Sta/Elev= 29
  4713.5  979.42  4719.5  978.91  4729.5  978.53  4739.5  977.57  4749.5  977.21
  4759.5  976.68  4765.9   975.6  4770.9  975.11  4799.6  973.74  4819.7  973.09
  4829.7   972.3  4839.7  970.17  4849.7  970.43  4995.5  969.38  4995.8  968.88
  4999.3  968.88  4999.5  969.38  5020.1  969.48  5180.8   969.4  5190.8  971.74
  5200.9     974  5210.9  975.05    5231  976.41  5251.1  978.02  5261.1  978.46
  5268.7  979.29  5273.7  979.58  5281.2  979.77  5287.8  979.79
#Mann= 3 ,-1 , 0
  4713.5     .05       0  4995.5    .033       0  4999.5     .05       0
Bank Sta=4995.5,4999.5
XS Rating Curve= 0 ,0
Exp/Cntr=0.3,0.1

Type RM Length L Ch R = 1 ,17414   ,44,44,44
BEGIN DESCRIPTION:
Miller Creek 39.3
END DESCRIPTION:
XS GIS Cut Line= 2
      2287963.33      7199986.96      2287429.24      7200082.66
#Sta/Elev= 30
  4761.9  981.15  4766.6  981.15  4786.6  979.37  4796.8   978.1  4809.8  977.26
  4817.1  976.38  4827.3  974.75  4837.4  973.76  4847.6  973.18  4857.7  970.65
  4863.5  969.91  4878.1  969.94  4888.2  969.55  4908.5  969.42    5000  969.54
  5018.3  969.38  5018.5  968.88    5022  968.88  5022.3  969.38  5162.5  969.84
  5172.7  970.77  5182.8  972.93    5193   972.9  5201.2  973.71  5206.3  973.34
  5233.6   974.4    5260  975.52  5274.3  976.71  5284.4  976.71  5304.5  977.23
#Mann= 3 ,-1 , 0
  4761.9     .05       0  5018.3    .033       0  5022.3     .05       0
Bank Sta=5018.3,5022.3
XS Rating Curve= 0 ,0
Exp/Cntr=0.3,0.1

Type RM Length L Ch R = 1 ,17370   ,111,111,111
BEGIN DESCRIPTION:
Miller Creek 39.2
END DESCRIPTION:
XS GIS Cut Line= 2
      2287936.09      7199947.02      2287402.68      7200049.68
#Sta/Elev= 30
  4769.8  980.61  4797.4  977.88  4807.2   975.5  4812.3  976.28  4817.8  974.14
  4827.9  973.33  4838.1  974.02  4864.3  973.86    4889  974.42  4968.1  973.82
  4990.9  974.38    5020  974.17  5031.6  974.66  5062.2  973.88  5071.9  973.18
    5077   974.1  5102.9  974.17  5123.3  972.87  5126.9  972.29  5127.2  971.79
  5130.7  971.79  5130.9  972.29    5134  974.61    5164  972.74  5180.8  972.94
  5185.9  973.54  5214.9  973.08  5255.6  975.52    5276  975.52    5313  977.43
#Mann= 3 ,-1 , 0
  4769.8     .05       0  5126.9    .033       0  5130.9     .05       0
Bank Sta=5126.9,5130.9
XS Rating Curve= 0 ,0
Exp/Cntr=0.3,0.1

Type RM Length L Ch R = 1 ,17259   ,155,155,155
BEGIN DESCRIPTION:
Miller Creek 39.1
END DESCRIPTION:
XS GIS Cut Line= 2
       2287894.3      7199854.63      2287432.66      7199955.81
#Sta/Elev= 30
  4730.5  979.31  4775.4  974.38  4780.5  974.59  4807.6  965.48  4824.3  965.68
  4829.4  966.33  4838.3  965.95  4848.5   967.1  4873.2  966.25  4879.3  965.01
  4899.7  963.99  4917.1  963.91  4922.2  964.74  4930.4  964.69  4960.9  963.31
  5009.8     962    5015  962.39  5051.3  961.68  5051.5  961.18    5055  961.18
  5055.3  961.68    5084  963.23  5107.7   966.8  5114.7  968.53  5124.9  970.22
  5135.2  971.15  5151.6  970.56  5176.1  972.35  5195.4  972.72  5203.1  973.62
#Mann= 3 ,-1 , 0
  4730.5     .05       0  5051.3    .033       0  5055.3     .05       0
Bank Sta=5051.3,5055.3
XS Rating Curve= 0 ,0
Exp/Cntr=0.3,0.1

Type RM Length L Ch R = 1 ,17104   ,296,296,296
BEGIN DESCRIPTION:
Miller Creek 39.0
END DESCRIPTION:
XS GIS Cut Line= 3
      2287877.35      7199645.58      2287556.53      7199783.07
      2287374.41      7199855.15
#Sta/Elev= 30
  4647.4  980.15  4672.1  975.97  4678.2  974.41  4689.1  973.22  4710.9  969.07
  4719.2  967.02  4732.6  965.39  4748.2  964.84  4795.4  961.53  4841.4   960.3
  4863.2  960.47  4871.5  959.71    4875  958.64  4875.2  958.14  4878.7  958.14
    4879  958.64    4885  960.02  4900.5  960.46  4982.9  960.39  4996.4  961.01
  5000.4  961.94  5005.8  961.86  5054.5  967.46  5059.9  967.17  5078.8  968.34
  5090.6  968.07  5101.3  969.24  5132.9  969.93    5168  971.83  5192.3  972.32
#Mann= 3 ,-1 , 0
  4647.4     .05       0    4875    .033       0    4879     .05       0
Bank Sta=4875,4879
XS Rating Curve= 0 ,0
Exp/Cntr=0.3,0.1

Type RM Length L Ch R = 1 ,16808   ,350,350,350
BEGIN DESCRIPTION:
Miller Creek 38.0
END DESCRIPTION:
XS GIS Cut Line= 3
      2287846.01      7199514.31      2287626.17      7199533.77
      2287335.36      7199574.16
#Sta/Elev= 30
  4782.6  977.89  4792.5  975.27  4799.7  974.01  4819.8  972.91  4839.8  973.01
  4849.9   972.2    4870  968.45    4880   967.2  4899.5  965.72  4910.1  963.94
  4940.2  960.98  4970.3  958.48  4980.4  958.26  4990.4  957.19  4997.4  954.49
  4997.6  953.99  5001.1  953.99  5001.4  954.49  5008.9  955.51  5013.9  954.78
  5020.6  956.59  5030.7  957.31  5040.8  957.17  5050.9  957.72  5101.4  957.47
  5157.3  958.16  5202.4  959.48    5229  961.01  5252.8  962.93  5296.9  963.39
#Mann= 3 ,-1 , 0
  4782.6     .05       0  4997.4    .033       0  5001.4     .05       0
Bank Sta=4997.4,5001.4
XS Rating Curve= 0 ,0
Exp/Cntr=0.3,0.1

Type RM Length L Ch R = 1 ,16458   ,361,361,361
BEGIN DESCRIPTION:
Miller Creek 37.0
END DESCRIPTION:
XS GIS Cut Line= 3
      2287584.04      7199026.83        2287429.        7199260.
      2287279.01      7199559.99
#Sta/Elev= 30
  4719.7  974.72  4754.7  972.22  4760.7  969.95  4769.7  968.73  4775.7  966.43
  4790.8  965.08  4796.8  963.81  4826.9   960.6  4832.9  959.36  4841.9  958.82
  4847.9  957.37  4862.9  956.31  4868.9  955.13    4905  953.56  4963.7  954.54
  4977.2  953.69  4990.2  951.62  4990.4  951.12  4993.9  951.12  4994.2  951.62
  4996.7  952.59  5002.5  952.59  5008.1  954.03  5133.9  954.14  5245.7  958.82
  5290.4  961.53  5298.8  961.57  5304.4  960.44  5312.8  963.01  5335.1  964.27
#Mann= 3 ,-1 , 0
  4719.7     .05       0  4990.2    .033       0  4994.2     .05       0
Bank Sta=4990.2,4994.2
XS Rating Curve= 0 ,0
Exp/Cntr=0.3,0.1

Type RM Length L Ch R = 1 ,16097   ,344,344,344
BEGIN DESCRIPTION:
Miller Creek 36.0
END DESCRIPTION:
XS GIS Cut Line= 4
      2287583.03      7198942.43      2287312.33      7198967.88
       2287298.5      7199080.29      2287029.04      7199209.98
#Sta/Elev= 30
  4686.1  974.86  4714.4  973.41  4730.3  970.23  4800.6  963.95  4810.7   962.4
    4818  959.88  4850.9  956.15  4921.2  952.54  4926.7  950.44  4931.7  949.78
  4941.2  951.89  4951.3  950.44  4955.2  949.08  4955.4  948.58  4958.9  948.58
  4959.2  949.08  4990.4  951.14  5025.9  951.45  5040.7  950.85  5079.2  951.17
  5092.9   951.7  5101.8  950.79  5115.1  950.45  5137.3  952.34  5197.9  953.57
  5220.5   954.9  5237.2  957.13  5259.4  958.83  5265.8  959.85  5370.3  965.79
#Mann= 3 ,-1 , 0
  4686.1     .05       0  4955.2    .033       0  4959.2     .05       0
Bank Sta=4955.2,4959.2
XS Rating Curve= 0 ,0
Exp/Cntr=0.3,0.1

Type RM Length L Ch R = 1 ,15753   ,313,313,313
BEGIN DESCRIPTION:
Miller Creek 35.0
END DESCRIPTION:
XS GIS Cut Line= 3
       2287572.5      7198907.69       2287180.3      7198918.94
      2286889.62      7198939.87
#Sta/Elev= 30
  4608.4   974.1  4631.9  972.92  4661.9  968.47  4671.9  967.84  4691.9  965.66
    4722  963.51    4732  961.07    4742  959.87    4772  957.51    4852  952.35
  4860.1  950.31  4865.1  949.69    4872   950.5    4882  949.87    4922  949.41
    4952  948.72  4972.1  947.73  4990.1  947.59  4990.3  947.09  4993.8  947.09
  4994.1  947.59  5022.1  947.69  5042.2  950.48  5052.2  952.83  5062.2  953.74
  5081.2  952.39  5092.3  953.47  5132.4  955.56  5242.7  959.45  5292.2  960.52
#Mann= 3 ,-1 , 0
  4608.4     .05       0  4990.1    .033       0  4994.1     .05       0
Bank Sta=4990.1,4994.1
XS Rating Curve= 0 ,0
Exp/Cntr=0.3,0.1

Type RM Length L Ch R = 1 ,15440   ,374,374,374
BEGIN DESCRIPTION:
Miller Creek 34.0
END DESCRIPTION:
XS GIS Cut Line= 3
        2287329.        7198560.        2287129.        7198660.
      2286978.99      7198760.01
#Sta/Elev= 30
    4781  959.49  4783.8  959.49  4789.4  957.51    4795  957.55  4811.7  950.94
  4825.7  948.77  4839.7   947.8  4870.4  947.58  4878.8  946.99  4959.9  947.21
  4982.2  946.77  4990.6  946.05  4999.8  941.83  5000.1  941.33  5003.6  941.33
  5003.8  941.83  5007.6  941.83  5012.1  943.66  5018.1   945.4  5027.1  945.38
  5033.1   946.1  5054.2  945.35  5063.2  945.47  5069.2  946.27  5120.3   944.5
  5135.3  949.19  5141.3  951.73  5156.3  956.64  5177.4  957.05  5184.9  956.73
#Mann= 3 ,-1 , 0
    4781     .05       0  4999.8    .033       0  5003.8     .05       0
Bank Sta=4999.8,5003.8
XS Rating Curve= 0 ,0
Exp/Cntr=0.3,0.1

Type RM Length L Ch R = 1 ,15066   ,335,335,335
BEGIN DESCRIPTION:
Miller Creek 33.0
END DESCRIPTION:
XS GIS Cut Line= 3
      2287279.04      7198209.98        2286979.        7198360.
      2286776.41      7198464.71
#Sta/Elev= 30
  4668.6  962.71    4691  959.31  4727.3  957.81  4744.1  952.78  4766.5  948.81
  4772.1  949.15  4788.8  946.64  4794.4  947.14  4833.6  942.39  4861.5  941.15
  4892.2  943.16    4923  942.32  4950.9  943.03  4959.3  941.43  4973.3  941.56
  4988.1  938.87  4988.3  938.37  4992.1  938.87  5006.9  939.71  5012.3  942.58
  5040.1  943.72  5078.8  947.47  5106.5  948.18  5116.6  949.02    5123  950.88
  5128.7  950.17  5145.2  953.72  5150.8  952.84  5167.3  954.79  5232.1  958.61
#Mann= 3 ,-1 , 0
  4668.6     .05       0  4988.1    .033       0  4992.1     .05       0
Bank Sta=4988.1,4992.1
XS Rating Curve= 0 ,0
Exp/Cntr=0.3,0.1

Type RM Length L Ch R = 1 ,14731   ,362,362,362
BEGIN DESCRIPTION:
Miller Creek 32.0
END DESCRIPTION:
XS GIS Cut Line= 3
        2287229.        7198060.        2287079.        7198060.
      2286847.38       7198082.3
#Sta/Elev= 30
  4850.1  955.78  4852.6  955.78  4860.1  954.96  4880.1  950.75  4890.1   950.2
  4900.1  946.72  4910.1  943.61  4920.1  942.88  4930.1  940.08  4940.1  939.44
  4950.1  939.42  4960.1  937.59  4968.1  936.65  4968.4  936.15  4971.9  936.15
  4972.1  936.65  4980.1  937.57  4990.1  940.28  5002.6  940.07  5040.3   938.4
  5048.8  938.93  5060.4  940.58  5070.4  941.26  5080.5   942.4  5090.5  942.75
  5110.6  944.53  5180.9  947.65    5191  949.16    5201  950.23  5232.8  951.92
#Mann= 3 ,-1 , 0
  4850.1     .05       0  4968.1    .033       0  4972.1     .05       0
Bank Sta=4968.1,4972.1
XS Rating Curve= 0 ,0
Exp/Cntr=0.3,0.1

Type RM Length L Ch R = 1 ,14369   ,347,347,347
BEGIN DESCRIPTION:
Miller Creek 31.0
END DESCRIPTION:
XS GIS Cut Line= 3
      2287129.04      7197759.99        2286929.        7197810.
      2286828.99        7197810.
#Sta/Elev= 30
  4798.9  954.59  4801.5  954.59    4817  942.56  4822.1   941.5  4829.9  938.83
  4840.2  936.81  4850.5  936.66  4871.1  937.02  4891.7  937.08  4899.4  937.32
  4922.6  937.39  4932.9  937.89  4940.7  937.56  4945.8  936.69  4964.6  935.46
  4974.2  935.98  4987.1  935.42  4994.8  934.71  5002.5  934.34  5007.6  934.34
  5013.1  932.64  5013.3  932.14  5016.8  932.14  5017.1  932.64  5025.1  934.37
  5035.1  939.51  5045.1  941.17  5055.1  943.25  5085.1  945.64  5105.1  946.35
#Mann= 4 ,-1 , 0
  4798.9     .12       0  4964.6     .05       0  5013.1    .033       0
  5017.1     .05       0
Bank Sta=5013.1,5017.1
XS Rating Curve= 0 ,0
Exp/Cntr=0.3,0.1

Type RM Length L Ch R = 1 ,14022   ,524,524,524
BEGIN DESCRIPTION:
Miller Creek 30.0
END DESCRIPTION:
XS GIS Cut Line= 3
      2287028.96        7197510.        2286879.        7197510.
      2286526.29      7197514.19
#Sta/Elev= 30
  4854.3  950.04  4856.8  950.04  4864.3  948.31  4874.3   944.5  4884.3   938.3
  4894.3   934.3  4904.3  933.52  4934.3  932.75  4944.3   932.7  4964.3  933.53
  4984.3  932.49  4994.3  932.61  5001.8  931.54  5007.1  931.48  5022.3   928.4
  5022.5   927.9    5026   927.9  5026.3   928.4  5034.3   933.9  5084.3  934.68
  5104.3  935.66  5114.3  935.65  5124.3  934.46  5154.3  936.64  5174.3  936.52
  5194.3  935.44  5234.3  939.71  5264.3  941.54  5304.3  944.45    5357  946.94
#Mann= 4 ,-1 , 0
  4854.3     .12       0  5007.1     .05       0  5022.3     .07       0
  5026.3     .05       0
Bank Sta=5022.3,5026.3
XS Rating Curve= 0 ,0
Exp/Cntr=0.3,0.1

Type RM Length L Ch R = 1 ,13498   ,198,198,198
BEGIN DESCRIPTION:
Miller Creek 29.0
END DESCRIPTION:
XS GIS Cut Line= 4
      2287178.99        7196860.      2286719.48      7197065.89
      2286682.78      7197288.47      2286497.68      7197464.13
#Sta/Elev= 30
  4401.1  953.56  4409.9  952.75  4415.4  950.89  4461.8  950.26  4477.8  949.09
    4485  946.71  4490.5  943.63  4543.5  940.96    4560  941.14  4566.6  939.37
  4606.4  936.35  4611.9  934.83  4629.6  935.56  4681.4  933.77  4802.8  930.56
  4969.6  929.85  4977.5   924.8  4977.9   924.3  4981.9   924.8  4989.9  925.11
  4997.4  927.23  5002.4  926.18  5010.1  927.77  5020.3  928.24  5091.2  928.21
    5135  930.57  5162.4  938.81  5169.3  943.22  5197.6  945.76  5385.4  949.32
#Mann= 5 ,-1 , 0
  4401.1     .05       0  4566.6     .12       0  4681.4     .05       0
  4977.5    .033       0  4981.9     .05       0
Bank Sta=4977.5,4981.9
XS Rating Curve= 0 ,0
Exp/Cntr=0.3,0.1

Type RM Length L Ch R = 1 ,13300   ,240,240,240
BEGIN DESCRIPTION:
Miller Creek 28.1
END DESCRIPTION:
XS GIS Cut Line= 2
      2286943.11      7196891.68      2286294.83      7197223.79
#Sta/Elev= 30
  4536.5  933.21  4589.7  933.18  4619.8  931.57  4650.7  931.54  4672.9  930.22
  4732.1  929.04  4754.6  930.02  4783.9  928.55  4806.1  928.23  4878.3  928.18
  4933.7  927.17  4961.5  927.88  4968.1  927.23  4978.1  924.16  4981.5  924.07
  4981.9  923.57  4985.5  923.57  4985.9  924.07  5000.3  925.49  5005.9  928.95
    5013  939.18  5022.5  945.33  5035.5  947.94  5066.9  949.57  5111.3  950.49
  5139.1  950.41  5177.9   953.1  5183.5  953.03  5244.5  956.31  5264.9  956.73
#Mann= 3 ,-1 , 0
  4536.5     .05       0  4981.5    .033       0  4985.9     .05       0
Bank Sta=4981.5,4985.9
XS Rating Curve= 0 ,0
Exp/Cntr=0.3,0.1

Type RM Length L Ch R = 1 ,13060   ,233,233,233
BEGIN DESCRIPTION:
Miller Creek 28.0
END DESCRIPTION:
XS GIS Cut Line= 3
      2286978.98        7196810.      2286704.95      7196883.93
      2286282.18      7196871.12
#Sta/Elev= 30
  4590.3  939.76  4621.4  937.81  4647.6   930.6  4652.7   930.9  4673.1  930.09
  4714.6  929.71  4727.4  930.26  4762.1  929.15  4796.8  928.87  4849.2  926.78
  4874.1  926.57  4880.1  925.91  4970.1   924.7  4987.9  923.06  4988.3  922.56
  4991.9  922.56  4992.3  923.06  5010.1  923.35  5020.1  925.31  5030.2  931.16
  5040.2  933.75  5060.2     940  5080.2  940.58  5110.2  939.89  5130.2  943.12
  5150.2  945.27  5172.1  946.42  5180.2  947.39  5210.2   948.8  5297.1  951.75
#Mann= 3 ,-1 , 0
  4590.3     .05       0  4987.9    .033       0  4992.3     .05       0
Bank Sta=4987.9,4992.3
XS Rating Curve= 0 ,0
Exp/Cntr=0.3,0.1

Type RM Length L Ch R = 1 ,12827   ,269,269,269
BEGIN DESCRIPTION:
Miller Creek 27.1
END DESCRIPTION:
XS GIS Cut Line= 2
       2287115.7      7196741.71      2286357.22      7196668.52
#Sta/Elev= 30
  4609.4  948.94  4636.2  948.56  4675.3  942.74  4680.3  943.32  4686.5  942.51
  4716.6  942.12  4726.6  940.81  4756.8   932.2  4776.9  931.24  4787.6  929.76
  4837.2  928.03  4957.7  927.04  5005.7  920.92  5006.1  920.42  5009.7  920.42
  5010.2  920.92    5018  921.07    5028  922.69  5048.1     923  5058.2   921.8
  5078.3  921.81  5094.5  925.25  5099.5  924.69  5108.4   926.2  5118.5  928.63
  5128.5  929.82  5158.6  936.31  5178.7  939.78    5229  940.94  5371.4  947.74
#Mann= 3 ,-1 , 0
  4609.4     .05       0  5005.7    .033       0  5010.2     .05       0
Bank Sta=5005.7,5010.2
XS Rating Curve= 0 ,0
Exp/Cntr=0.3,0.1

Type RM Length L Ch R = 1 ,12558   ,72,72,72
BEGIN DESCRIPTION:
Miller Creek 27.0
END DESCRIPTION:
XS GIS Cut Line= 6
      2287084.37      7196588.11      2286820.62      7196531.81
      2286776.45      7196446.53      2286716.35      7196355.89
      2286587.88      7196276.69      2286454.35      7196268.44
#Sta/Elev= 30
  4639.6  949.67  4652.4  946.66  4657.5  946.32  4665.5  941.87    4686  939.86
  4701.9  936.91  4746.3  931.18  4751.4  931.49  4795.8  927.74  4800.9  928.12
  4839.4  926.25  4859.8  924.51  4889.7  925.28  4900.7  924.45  4913.1  924.63
  4942.5   922.9  4990.1  917.86  4990.6  917.36  4994.6  917.86  5023.5  918.76
  5029.5  920.63  5044.6  920.12  5065.6  921.44  5080.7  920.95  5086.7  922.01
  5116.3  921.88  5216.8  926.18    5324  933.23  5364.1  936.98  5398.8  938.45
#Mann= 3 ,-1 , 0
  4639.6     .05       0  4990.1    .033       0  4994.6     .05       0
Bank Sta=4990.1,4994.6
XS Rating Curve= 0 ,0
Exp/Cntr=0.3,0.1

Type RM Length L Ch R = 1 ,12486   ,228,228,228
BEGIN DESCRIPTION:
Miller Creek 26.1
END DESCRIPTION:
XS GIS Cut Line= 6
      2287128.52      7196533.15      2286847.26      7196481.86
      2286833.72      7196419.39      2286738.48      7196321.48
      2286603.13      7196204.12      2286455.02      7196200.92
#Sta/Elev= 30
  4604.9  951.77  4634.9   949.3  4645.1   945.6  4650.2  942.81  4655.3  942.08
  4695.9  939.84  4703.5  937.74  4708.6  938.32  4807.7  928.41  4820.3  928.11
  4887.4  922.96  4894.3  922.96  4913.2  920.46  4923.4  920.44  4943.9  921.73
  4957.8   920.3  4978.9  918.57  4984.1  917.46  5021.3   918.4  5028.3  919.47
  5134.3  921.94    5170  923.35  5177.1  924.23  5183.7  923.78  5248.3  927.13
    5255  926.96  5269.2  929.52  5284.6  930.47  5324.6  935.76  5418.6  939.18
#Mann= 3 , 0 , 0
  4604.9     .05       0  4957.8    .033       0  5028.3     .05       0
Bank Sta=4957.8,5028.3
XS Rating Curve= 0 ,0
Exp/Cntr=0.3,0.1

Type RM Length L Ch R = 1 ,12258   ,308,308,308
BEGIN DESCRIPTION:
Miller Creek 26.0
END DESCRIPTION:
XS GIS Cut Line= 3
      2287044.55      7196208.49      2286831.49      7196168.29
      2286502.46      7196111.59
#Sta/Elev= 30
  4782.4  946.65    4788  943.95  4797.2  942.64  4802.3  943.52  4818.6  941.33
  4849.1  933.73  4854.7  931.21  4859.8   931.2  4889.8  925.84    4900  924.86
  4912.2   922.2  4920.3  919.54  4964.6  914.88  4979.6  911.78  4983.2  911.78
  4991.6  916.11  4997.9  917.98  5032.2  917.53  5052.5   917.9  5072.6  918.84
  5077.7  919.64  5113.4  920.23  5174.3  923.44  5184.4  924.87  5192.4  926.84
  5197.4  926.51  5204.7  929.02    5225  934.34  5235.1  935.45  5333.1  939.27
#Mann= 3 , 0 , 0
  4782.4     .05       0  4920.3    .033       0  4997.9     .05       0
#XS Ineff= 2 , 0
       0                  5011.9       0  918.22
Permanent Ineff=
       F       F
Bank Sta=4920.3,4997.9
XS Rating Curve= 0 ,0
Exp/Cntr=0.3,0.1

Type RM Length L Ch R = 1 ,11950   ,177,177,177
BEGIN DESCRIPTION:
Miller Creek 25.1
END DESCRIPTION:
XS GIS Cut Line= 3
      2287118.37      7195846.26       2286884.9      7195946.33
      2286593.23        7196073.
#Sta/Elev= 30
    4808  958.51  4832.4  957.96  4850.5  955.96  4855.9  956.26  4861.7   952.4
  4872.6  948.24  4879.5  946.67  4908.5  942.42  4916.1  940.48  4926.6  940.18
  4937.9   935.2  4948.8  929.28  4955.6  922.61  4968.7  907.32  4972.3  907.32
  4979.2  909.18  4984.7   911.8  4992.3  913.15  5024.9   915.8  5068.4  916.37
  5101.2  915.29  5144.8  915.66  5177.5  917.76  5221.1  917.97  5275.6  920.29
  5288.3  921.22  5329.7  927.46  5335.2     927  5358.6  934.67    5380  936.05
#Mann= 3 , 0 , 0
    4808     .05       0  4955.6    .033       0  4992.3     .05       0
#XS Ineff= 2 , 0
       0                  5068.4       0  916.37
Permanent Ineff=
       F       F
Bank Sta=4955.6,4992.3
XS Rating Curve= 0 ,0
Exp/Cntr=0.3,0.1

Type RM Length L Ch R = 1 ,11773   ,215,215,215
BEGIN DESCRIPTION:
Miller Creek 25.0
END DESCRIPTION:
XS GIS Cut Line= 3
      2286856.93      7195655.99      2286769.01      7195917.04
      2286579.04      7196059.97
#Sta/Elev= 30
  4784.5  946.06  4793.9  946.26  4820.1  943.41  4825.3  944.14  4830.9  942.24
  4852.3  938.06  4856.8   940.8  4883.1  928.27  4888.3  929.33  4894.3  926.35
  4914.5  919.88  4919.8  921.71  4925.9  917.44  4936.5  915.16  4947.1  914.73
  4957.6  912.11  4968.1  911.04  4982.8   908.3  4987.4  906.66  5014.3  909.83
  5020.9  912.32  5058.9  915.91    5076  916.68    5126  917.85  5140.5  917.39
  5203.9  923.82  5225.9  928.43  5247.7  929.47  5275.9  934.95  5297.7  936.19
#Mann= 5 ,-1 , 0
  4784.5     .05       0  4852.3     .12       0  4947.1     .05       0
  4957.6    .033       0  5020.9     .05       0
Bank Sta=4957.6,5020.9
XS Rating Curve= 0 ,0
Exp/Cntr=0.3,0.1

Type RM Length L Ch R = 1 ,11558   ,233,233,233
BEGIN DESCRIPTION:
Miller Creek 24.1
END DESCRIPTION:
XS GIS Cut Line= 3
      2286802.25      7195640.31       2286634.9      7195725.32
      2286463.11      7195986.95
#Sta/Elev= 30
  4746.7  946.84    4787   946.1  4817.6  945.58  4823.3  945.02  4828.9  942.96
  4839.9  942.65  4845.5   938.9  4862.2  937.82  4867.8  932.49  4884.4  931.61
    4890  928.27  4906.7  927.08  4912.3  923.42    4929  921.56  4934.1  916.11
  4950.1  914.58  4963.9   914.3  4992.3  908.29  4999.8  905.36  5009.4  904.74
    5011  904.73  5011.5  904.23  5015.6  904.73  5049.5  911.36  5064.6  912.61
  5079.7  915.16  5107.5  917.72    5131  920.95  5194.2  932.92  5247.4   935.9
#Mann= 5 ,-1 , 0
  4746.7     .05       0    4787     .12       0  5009.4     .05       0
    5011     .07       0  5015.6     .05       0
Bank Sta=5011,5015.6
XS Rating Curve= 0 ,0
Exp/Cntr=0.3,0.1

Type RM Length L Ch R = 1 ,11325   ,278,278,278
BEGIN DESCRIPTION:
Miller Creek 24.0
END DESCRIPTION:
XS GIS Cut Line= 3
      2286628.98      7195610.01        2286429.        7195660.
      2286159.27      7195711.86
#Sta/Elev= 30
  4793.7  937.86  4796.3  937.86  4811.7  929.58  4834.9  924.91  4852.9  917.48
  4876.1  911.96  4907.1  908.82  4948.3  907.47  4981.8  907.96  5002.4  906.18
    5010  903.77  5023.5  903.61    5024  903.11  5028.1  903.61  5040.6  906.67
  5060.9  908.82  5077.7  908.59  5120.5  911.34  5162.8  918.75  5172.9  918.05
  5181.6  914.68  5186.7  916.22  5193.3  912.68  5203.5  913.65  5213.7  920.07
  5223.9  922.58  5238.7  923.74  5244.2  925.77  5264.6  928.16  5274.5   930.5
#Mann= 4 ,-1 , 0
  4793.7     .12       0  5023.5     .07       0  5028.1     .12       0
  5120.5     .05       0
Bank Sta=5023.5,5028.1
XS Rating Curve= 0 ,0
Exp/Cntr=0.3,0.1

Type RM Length L Ch R = 1 ,11047   ,377,377,377
BEGIN DESCRIPTION:
Miller Creek 23.1
END DESCRIPTION:
XS GIS Cut Line= 2
      2286801.35      7195397.89      2286014.82      7195450.69
#Sta/Elev= 30
  4526.2  942.68  4548.6   938.3  4568.6  929.69  4578.7  927.48  4598.7   924.2
    4632  921.28  4648.8  918.92  4688.9  918.23  4749.1  914.32  4777.9  908.19
  4782.9  912.18  4789.1  913.09  4839.3  908.55  4909.4  905.32  4949.5  905.75
  4977.2  898.76  4977.7  898.26  4981.9  898.76  4999.6  902.92  5009.6  903.54
  5029.7   913.3  5039.7  916.03  5049.7  917.83  5068.9  918.39  5099.8  917.55
  5129.9  913.02    5160  917.55    5180  923.69  5210.1  927.33  5314.5  931.33
#Mann= 5 ,-1 , 0
  4526.2     .05       0    4632     .12       0  4977.2     .07       0
  4981.9     .12       0  5068.9     .05       0
Bank Sta=4977.2,4981.9
XS Rating Curve= 0 ,0
Exp/Cntr=0.3,0.1

Type RM Length L Ch R = 1 ,10670   ,298,298,298
BEGIN DESCRIPTION:
Miller Creek 23.0
END DESCRIPTION:
XS GIS Cut Line= 3
      2286683.12      7195240.86      2286513.08      7195180.74
      2286272.98      7195141.71
#Sta/Elev= 30
  4816.5  938.86  4821.3  938.86  4830.1  933.82  4834.1  934.16  4842.1   931.2
    4861  927.04  4866.3  927.13  4884.5  918.74  4891.9  913.07  4897.3  914.61
  4905.7  909.79  4922.9   907.2  4969.4  905.95  4984.7  901.56  4988.2   896.6
  4988.7   896.1    4993   896.6  4996.4  897.58  5001.4  897.58  5021.2  901.62
  5041.5  901.51    5091   903.4  5096.1  902.87  5112.4  903.66  5142.8  903.45
  5157.7  904.67  5183.3  914.83  5213.7  924.98  5224.3  925.07  5240.1  927.55
#Mann= 3 ,-1 , 0
  4816.5     .12       0  4988.2     .07       0    4993     .12       0
Bank Sta=4988.2,4993
XS Rating Curve= 0 ,0
Exp/Cntr=0.3,0.1

Type RM Length L Ch R = 1 ,10372   ,242,242,242
BEGIN DESCRIPTION:
Miller Creek 22.0
END DESCRIPTION:
XS GIS Cut Line= 3
      2286528.99      7194810.01      2286439.38       7194924.6
      2286279.01      7195109.99
#Sta/Elev= 30
  4857.1  944.42  4860.3  944.42  4864.3  941.33  4893.2  929.75  4899.6  928.81
  4907.7  925.35  4914.1  923.85  4920.6   918.2  4928.5  913.31  4934.9  912.49
    4943  909.54  4949.3  909.06  4957.5  906.03  4984.6  899.82  4992.7  896.93
  5011.1  894.05  5011.7  893.55    5016  894.05  5021.2  895.55  5027.8   895.5
  5035.5  898.24  5042.1  899.19  5134.2  901.02  5162.7  904.46  5212.1  908.48
  5226.3  911.44    5234  914.41  5240.6  917.71  5244.4  922.74  5247.7  922.74
#Mann= 3 ,-1 , 0
  4857.1     .12       0  5011.1     .07       0    5016     .12       0
Bank Sta=5011.1,5016
XS Rating Curve= 0 ,0
Exp/Cntr=0.3,0.1

Type RM Length L Ch R = 1 ,10130   ,169,169,169
BEGIN DESCRIPTION:
Miller Creek 21.1
END DESCRIPTION:
XS GIS Cut Line= 3
      2286374.51      7194617.42      2286225.74      7194853.86
      2286156.66      7195090.32
#Sta/Elev= 30
  4791.4  937.26  4805.7  930.99  4818.1  928.27  4848.1  924.14  4854.1  919.67
  4863.4  918.84  4869.4  915.82  4884.6  914.56  4899.9  912.16  4905.9  910.36
  4921.1  908.94  4927.1  907.48  4957.6   905.6  4971.7   902.5  4997.6   893.3
  4998.2   892.8  5002.5   893.3  5007.1  895.23  5051.9  899.04  5087.6  898.93
  5118.8  897.37  5129.2  897.86  5160.5  903.23  5202.2   903.8  5257.4  907.32
  5285.5  914.09  5290.8  918.24    5296  919.65  5306.3  924.59  5317.1  925.82
#Mann= 3 ,-1 , 0
  4791.4     .12       0  4997.6     .07       0  5002.5     .12       0
Bank Sta=4997.6,5002.5
XS Rating Curve= 0 ,0
Exp/Cntr=0.3,0.1

Type RM Length L Ch R = 1 ,9961    ,450,450,450
BEGIN DESCRIPTION:
Miller Creek 21.0
END DESCRIPTION:
XS GIS Cut Line= 3
      2286329.01      7194559.99      2286130.85      7194731.07
        2286079.      7195060.02
#Sta/Elev= 30
  4658.4  943.47  4661.7  943.47  4672.1  936.83  4679.8  933.78  4708.3  928.23
  4750.9  910.44  4771.9  905.92  4821.3  901.65  4843.2   900.5  4864.1  900.83
  4870.7   897.7  4884.9  894.56  4913.5  896.74  4964.4  896.37  4987.5  891.11
  4988.1  890.61  4992.4  891.11  5000.1  891.38  5020.3  895.69  5060.8  894.47
  5089.4  899.52  5151.9  904.88  5182.3   906.4  5202.6  909.62  5212.7  913.09
  5219.4   917.6  5224.5  917.94  5243.1  925.52  5248.3  925.87  5253.2  926.03
#Mann= 4 ,-1 , 0
  4658.4     .12       0  4987.5     .07       0  4992.4     .12       0
  5248.3     .05       0
Bank Sta=4987.5,4992.4
XS Rating Curve= 0 ,0
Exp/Cntr=0.3,0.1

Type RM Length L Ch R = 1 ,9511    ,392,392,392
BEGIN DESCRIPTION:
Miller Creek 20.0
END DESCRIPTION:
XS GIS Cut Line= 4
      2286276.47      7194505.26      2286041.12      7194626.29
      2285833.09      7194550.63       2285548.4      7194697.18
#Sta/Elev= 30
  4615.9  942.49  4639.2   934.5  4677.9  928.66  4683.5  925.34  4700.1  922.45
  4727.9  907.55  4766.6  898.29    4811  898.16  4833.2   895.1  4967.3  891.46
  4978.6  887.57  4995.5  885.83  4996.1  885.33  5000.4  885.83  5010.5  894.64
  5021.1  897.99  5111.8  897.77  5192.7  901.91  5305.7  911.34  5311.3  913.53
  5327.9  912.89  5333.5  916.59  5350.1  915.88  5355.7  918.84  5372.2  916.92
  5377.8  919.55  5394.4  918.62    5400  922.19  5416.6  920.76  5422.1  922.49
#Mann= 4 ,-1 , 0
  4615.9     .12       0  4995.5     .07       0  5000.4     .12       0
  5192.7     .05       0
Bank Sta=4995.5,5000.4
XS Rating Curve= 0 ,0
Exp/Cntr=0.3,0.1

Type RM Length L Ch R = 1 ,9119    ,199,199,199
BEGIN DESCRIPTION:
Miller Creek 19.0
END DESCRIPTION:
XS GIS Cut Line= 3
      2286066.25      7194286.71        2285879.        7194310.
       2285403.4      7194550.42
#Sta/Elev= 30
  4811.3   929.5  4848.8  923.49  4858.9  918.84  4876.2  914.87  4881.3   910.9
  4889.1   908.2  4919.4  900.25  4929.4  895.05  4949.6  889.05  4962.1  886.52
  4969.8  887.69  4979.8  886.16    4995  881.97  4995.6  881.47    5000  881.97
  5013.9  884.77  5022.4  891.59  5030.6  892.63  5075.2  891.72  5103.1  895.29
  5142.1  894.49  5156.9   892.3  5169.9  894.54  5186.6  892.48  5192.2  893.94
  5242.4  895.78  5370.5  903.65  5459.7  906.98    5493  905.76  5532.9  909.11
#Mann= 4 ,-1 , 0
  4811.3     .12       0    4995     .07       0    5000     .12       0
  5242.4     .05       0
Bank Sta=4995,5000
XS Rating Curve= 0 ,0
Exp/Cntr=0.3,0.1

Type RM Length L Ch R = 1 ,8920    ,250,250,250
BEGIN DESCRIPTION:
Miller Creek 18.1
END DESCRIPTION:
XS GIS Cut Line= 2
      2285925.51      7194032.88      2285371.37      7194526.04
#Sta/Elev= 30
  4770.9  935.32  4818.2  933.31  4865.5  930.87  4893.9  928.09  4908.1  925.46
    4929  916.33  4943.2  907.01    4965  895.83  4979.2  892.59  4993.4  885.35
  4997.6  880.91  4998.3  880.41  5002.6  880.91    5021  882.25  5035.2  887.65
  5049.4  888.18  5071.2   886.4  5077.9  888.16  5092.1  888.68  5099.6  891.17
  5106.3  892.24  5163.2  895.43  5237.3  897.75  5297.8  900.87  5318.7  900.71
  5354.6  903.44  5382.2  904.12  5481.7  909.45  5495.9  911.21  5512.7  911.58
#Mann= 5 ,-1 , 0
  4770.9     .05       0  4818.2     .12       0  4997.6     .07       0
  5002.6     .12       0  5237.3     .05       0
Bank Sta=4997.6,5002.6
XS Rating Curve= 0 ,0
Exp/Cntr=0.3,0.1

Type RM Length L Ch R = 1 ,8670    ,197,197,197
BEGIN DESCRIPTION:
Miller Creek 18.0
END DESCRIPTION:
XS GIS Cut Line= 3
        2285779.        7194010.        2285579.        7194060.
      2285278.97      7194210.01
#Sta/Elev= 30
  4792.9  927.38  4795.5  927.38  4810.9  918.72  4816.1  917.66  4834.1  907.55
  4865.1  894.42  4885.7  891.07  4893.4   888.2  4906.3  886.73  4916.6  887.21
  4934.6  885.81  4939.8   886.6  4986.2  878.75  4986.8  878.25  4991.2  878.75
  4996.5  885.03  5001.9  885.03  5007.4  891.06  5043.8  892.15  5096.9   890.9
  5176.9  896.17  5186.3  896.76  5200.3  899.52  5214.3  899.46    5245  903.08
    5259  909.06  5275.8  919.01  5281.4  918.85  5289.7  921.79  5334.5  925.37
#Mann= 4 ,-1 , 0
  4792.9     .12       0  4986.2     .07       0  4991.2     .12       0
  5176.9     .05       0
Bank Sta=4986.2,4991.2
XS Rating Curve= 0 ,0
Exp/Cntr=0.3,0.1

Type RM Length L Ch R = 1 ,8473    ,386,386,386
BEGIN DESCRIPTION:
Miller Creek 17.2
END DESCRIPTION:
XS GIS Cut Line= 2
      2285768.72      7193764.56      2285229.44      7194168.36
#Sta/Elev= 30
  4796.6  929.92  4830.7  929.01  4871.2  927.54  4885.3  928.87  4899.9   926.2
  4943.7  902.54  4979.1  888.73  4985.4  881.61  4991.2  878.05  4991.8  877.55
  4996.2  878.05  5021.1  878.44    5050  888.17  5064.6  890.19  5114.6  888.18
  5135.4  889.36    5171  886.08  5185.4  886.21  5285.4  896.91  5300.3  897.39
  5314.6   897.6  5393.8  905.82  5400.1  909.48  5414.6  909.43  5420.9  912.33
  5429.2  912.95  5435.5  919.15  5443.8  919.53  5450.1  922.14  5470.3  925.47
#Mann= 5 ,-1 , 0
  4796.6     .05       0  4830.7     .12       0  4991.2     .07       0
  4996.2     .12       0  5300.3     .05       0
Bank Sta=4991.2,4996.2
XS Rating Curve= 0 ,0
Exp/Cntr=0.3,0.1

Type RM Length L Ch R = 1 ,8087    ,337,337,337
BEGIN DESCRIPTION:
Miller Creek 17.1
END DESCRIPTION:
XS GIS Cut Line= 4
      2285580.13      7193599.79      2285311.77      7193796.42
      2285338.34      7193977.09      2284889.33      7194048.82
#Sta/Elev= 30
  4555.8  928.13  4578.7  927.21  4593.3   922.7  4606.8  915.42  4620.4  905.83
  4643.5  895.81  4664.4  890.43  4699.9  888.24  4850.4   886.1  4905.5  886.31
  4942.6   883.3  4962.9  879.02  4970.2  875.91  4980.5  874.45  4981.2  873.95
  4985.6  874.45  4993.2   876.8  5003.3  884.53  5013.4  887.19  5033.6   894.9
    5040  894.48    5045  892.73  5106.7  897.17  5180.7  900.29  5232.5  906.74
  5242.6  908.86  5247.8  912.66  5283.1  922.95    5315  926.58  5525.8  933.42
#Mann= 4 ,-1 , 0
  4555.8     .12       0  4980.5     .07       0  4985.6     .12       0
  5106.7     .05       0
Bank Sta=4980.5,4985.6
XS Rating Curve= 0 ,0
Exp/Cntr=0.3,0.1

Type RM Length L Ch R = 1 ,7750    ,451,451,451
BEGIN DESCRIPTION:
Miller Creek 17.0
END DESCRIPTION:
XS GIS Cut Line= 3
      2285501.66       7193551.7        2285179.        7193660.
      2284971.63      7193726.11
#Sta/Elev= 30
  4659.2  925.41  4663.2  925.41  4683.1  915.64  4705.2  901.91  4725.3  894.16
  4736.8  891.44  4794.6  886.47  4841.3  884.41  4904.6  884.21  4920.7   880.3
    4926  881.39  4936.3  879.93  4952.2  879.75  5002.2  881.05  5013.1  873.24
  5013.8  872.74  5018.2  873.24    5031  873.44  5041.5  875.89  5047.9  887.04
  5053.1  886.45  5062.5  890.08  5097.9   893.7  5112.3  894.64    5136  900.32
  5144.5  904.48  5149.7  905.81  5167.5  914.76  5188.5  920.73  5217.2  923.31
#Mann= 4 ,-1 , 0
  4659.2     .12       0  5013.1     .07       0  5018.2     .12       0
  5097.9     .05       0
Bank Sta=5013.1,5018.2
XS Rating Curve= 0 ,0
Exp/Cntr=0.3,0.1

Type RM Length L Ch R = 1 ,7299    ,247,247,247
BEGIN DESCRIPTION:
Miller Creek 16.0
END DESCRIPTION:
XS GIS Cut Line= 3
      2285429.04      7193310.01      2285185.13       7193247.7
      2284728.98      7193710.02
#Sta/Elev= 30
  4664.2   921.8  4674.6   921.1  4682.1  916.05  4687.2  916.04  4705.5  908.98
  4722.9  899.71  4746.8   893.7  4804.6  889.04  4845.5  888.81  4850.6  890.23
  4886.3  884.09  4921.9  881.49  4978.4  882.02  4992.6  880.29  4999.7  874.15
  5011.3  870.44  5011.9  869.94  5016.4  870.44    5028   870.8    5035  872.78
  5042.1  878.82  5056.3  881.24  5063.3  878.63  5070.4  880.42  5248.6  891.28
  5452.3  906.88  5515.9  916.49    5523  920.36  5537.1  923.14  5565.4  925.85
#Mann= 4 ,-1 , 0
  4664.2     .12       0  5011.3     .07       0  5016.4     .12       0
  5248.6     .05       0
Bank Sta=5011.3,5016.4
XS Rating Curve= 0 ,0
Exp/Cntr=0.3,0.1

Type RM Length L Ch R = 1 ,7052    ,210,210,210
BEGIN DESCRIPTION:
Miller Creek 15.1
END DESCRIPTION:
XS GIS Cut Line= 3
      2285426.02      7193257.08       2285131.1      7193092.34
        2284667.      7193641.62
#Sta/Elev= 30
  4710.5  921.71  4773.2  898.61  4919.4   890.9  4941.1  872.69  4947.6  871.31
  5000.5  869.76  5006.2  872.96  5027.9  876.39  5090.7  879.94  5097.6  879.61
    5105  875.08  5111.5  876.05  5119.3  869.82  5125.8  874.52  5133.6  869.54
  5166.1  869.24  5166.8  868.74  5171.2  869.24  5197.3  869.69  5203.8  873.58
  5211.6  871.77  5218.1  877.75  5225.9  877.77  5232.4  882.25  5324.7  883.32
  5424.2  889.83  5630.2   905.8  5658.8   912.4  5679.6  920.75  5767.4  927.91
#Mann= 4 ,-1 , 0
  4710.5     .12       0  5166.1     .07       0  5171.2     .12       0
  5424.2     .05       0
Bank Sta=5166.1,5171.2
XS Rating Curve= 0 ,0
Exp/Cntr=0.3,0.1

Type RM Length L Ch R = 1 ,6842    ,172,172,172
BEGIN DESCRIPTION:
Miller Creek 15.0
END DESCRIPTION:
XS GIS Cut Line= 3
      2285424.66      7192453.09      2285153.59      7192985.49
       2284634.9      7193585.01
#Sta/Elev= 30
    4403  918.27  4465.9  896.28    4523   888.6    4725  883.73  4747.4   881.1
  4760.7  875.73  4777.3  874.28  4782.9  870.65  4805.2  869.55  4821.8  869.58
  4827.4  872.19    4844   872.9  4849.6  876.73  4866.3  877.32  4894.1  882.34
  4955.2   883.9  4971.8  880.75  4977.5  875.44  4995.6  867.81  4996.8  867.31
  5003.9  867.81  5049.2   874.7  5063.4  873.84  5085.3  878.59  5233.4  882.19
  5333.2     882    5453  889.12  5687.5  910.24  5736.9  924.57  5793.2  928.43
#Mann= 4 ,-1 , 0
    4403     .12       0  4995.6     .07       0  5003.9     .12       0
    5453     .05       0
Bank Sta=4995.6,5003.9
XS Rating Curve= 0 ,0
Exp/Cntr=0.3,0.1

Type RM Length L Ch R = 1 ,6670    ,200,200,200
BEGIN DESCRIPTION:
Miller Creek 14.1
END DESCRIPTION:
XS GIS Cut Line= 4
      2285259.53      7192417.26      2285031.81      7192731.83
        2284998.       7193030.2      2284606.09       7193554.5
#Sta/Elev= 30
    4433  918.46  4448.7  917.12  4457.2  909.91  4492.8  896.67    4543  887.79
  4649.7  879.76    4708  881.02  4757.4  877.13  4839.6  875.71    4916  866.61
  4917.2  866.11  4924.3  866.61  4930.2  873.64  4940.3  878.39  4970.5  868.14
  4982.5  866.66  5030.8  873.65  5134.2  873.18  5157.1  879.51  5198.8  877.85
    5228  880.81  5313.5  881.69  5417.2   888.4  5478.1   893.5    5499  898.87
  5507.3  896.72  5628.2  905.36  5684.5  914.37  5728.2  925.94  5776.2  928.41
#Mann= 4 ,-1 , 0
    4433     .12       0    4916     .07       0  4924.3     .12       0
  5417.2     .05       0
Bank Sta=4916,4924.3
XS Rating Curve= 0 ,0
Exp/Cntr=0.3,0.1

Type RM Length L Ch R = 1 ,6470    ,545,545,545
BEGIN DESCRIPTION:
Miller Creek 14.0
END DESCRIPTION:
XS GIS Cut Line= 4
      2285102.87      7192385.01      2284834.62      7192855.07
      2284821.84      7193034.95      2284562.93      7193437.65
#Sta/Elev= 30
  4354.1   920.1  4368.8  913.47  4374.6  914.22  4382.9  909.47  4405.9  904.95
    4412  900.45  4433.6  896.33  4449.4   889.2  4514.3  877.05  4594.9  871.18
  4669.8  870.81    4693   866.3  4694.2   865.8  4701.3   866.3    4713   867.7
  4740.4  879.61  4762.8  880.63  4920.3  879.11  4940.4  876.33  4960.4   868.4
  5000.5   866.5  5060.7  876.87  5224.9   881.8  5245.4  889.71  5261.2  901.32
  5276.4  905.57  5421.7  908.39  5494.4  917.03  5515.5  923.54  5554.4  927.03
#Mann= 4 ,-1 , 0
  4354.1     .12       0    4693     .07       0  4701.3     .12       0
  5245.4     .05       0
Bank Sta=4693,4701.3
XS Rating Curve= 0 ,0
Exp/Cntr=0.3,0.1

Type RM Length L Ch R = 1 ,5925    ,369,369,369
BEGIN DESCRIPTION:
Miller Creek 13.0
END DESCRIPTION:
XS GIS Cut Line= 4
      2285005.33      7192332.13      2284781.36      7192732.47
      2284600.72       7192712.5        2284479.      7193110.01
#Sta/Elev= 30
  4438.4  921.59  4457.4  920.74  4500.8  907.38  4516.2  897.96  4522.5  886.45
  4528.2  885.41  4565.9   866.4  4609.3  866.33  4684.6  873.93  4802.6  880.11
  4907.1  876.56  4929.7  873.05  4949.8  867.04  4990.1  866.24    5006  866.09
  5007.2  865.59  5014.3  866.09  5030.3  866.42  5055.8  872.46  5096.9  876.82
  5128.5  876.67  5212.2  881.49  5243.6  885.47  5341.9  889.73  5412.7   896.3
  5445.4  904.57  5452.8  909.75    5473  917.04  5484.1  922.12  5494.6  922.64
#Mann= 6 ,-1 , 0
  4438.4     .12       0  4907.1     .05       0  4990.1     .12       0
    5006     .07       0  5014.3     .12       0    5473     .05       0
Bank Sta=5006,5014.3
XS Rating Curve= 0 ,0
Exp/Cntr=0.3,0.1

Type RM Length L Ch R = 1 ,5556    ,217,217,217
BEGIN DESCRIPTION:
Miller Creek 12.0
END DESCRIPTION:
XS GIS Cut Line= 3
      2284856.41      7191972.16      2284615.94       7192273.7
      2284405.48      7193069.04
#Sta/Elev= 30
  4421.1   914.6  4431.2  915.14  4439.3  911.76  4460.1  909.95  4468.1  905.02
  4474.5  906.52  4482.3  900.33  4538.5  893.23  4546.2  889.57  4695.5  879.92
  4738.1  881.87    4774  876.86  4780.3  878.12  4788.4  871.79  4835.3  866.63
  4852.4  866.24  4853.6  865.74    4861  866.24  4885.7  875.09  4906.4  867.45
  4916.7  866.25  5124.2  866.59  5154.7  871.89    5163  875.78  5283.7  877.66
  5392.6  883.07    5570  897.78  5589.1   901.1  5595.2  906.07  5629.5  921.59
#Mann= 6 ,-1 , 0
  4421.1     .12       0  4835.3     .05       0  4852.4    .033       0
    4861     .05       0  5124.2     .12       0    5570     .05       0
Bank Sta=4852.4,4861
XS Rating Curve= 0 ,0
Exp/Cntr=0.3,0.1

Type RM Length L Ch R = 1 ,5339    ,179,179,179
BEGIN DESCRIPTION:
Miller Creek 11.1
END DESCRIPTION:
XS GIS Cut Line= 3
      2284490.73      7192071.05      2284334.27      7192620.12
      2283396.65      7194622.99
#Sta/Elev= 30
  4543.5  925.92  4602.1  918.35  4680.2  883.02  4798.6  874.89  4943.6  866.17
  4944.9  865.67  4952.3  866.17  5072.7  866.93  5097.8  873.77  5378.6  888.38
  5704.9   908.4  5796.2  926.15  5870.2  917.51  5893.1  923.31  5921.4   917.2
  5938.7  924.52  5989.9  916.16  6007.2  921.79  6035.6  914.82  6058.4  925.38
  6109.6  911.34  6149.8  915.44  6231.1  906.09  6463.2  895.01  6737.2  896.73
  6759.5  885.29  6951.8  900.03  7164.8  913.42  7261.6   931.9  7325.9  933.89
#Mann= 8 ,-1 , 0
  4543.5     .12       0  4798.6     .05       0  4943.6    .033       0
  4952.3     .05       0  5097.8     .12       0  5378.6     .05       0
  6231.1     .12       0  6951.8     .05       0
#XS Ineff= 2 , 0
       0                  6074.9       0  924.05
Permanent Ineff=
       F       F
Bank Sta=4943.6,4952.3
XS Rating Curve= 0 ,0
Exp/Cntr=0.3,0.1
