--- Catlett Creek.prj (project) ---

Proj Title=Catlett Creek Base Level Engineering
Current Plan=p01
Default Exp/Contr=0.3,0.1
English Units
Geom File=g01
Flow File=f01
Plan File=p01
BEGIN DESCRIPTION:
Catlett Creek
END DESCRIPTION:

--- Catlett Creek.p01 (plan) ---

Plan Title=Multiple Run
Short Identifier=Multiple
Geom File=g01
Flow File=f01
Subcritical Flow
K Sum by GR= 0
Std Step Tol= 0.01
Critical Tol= 0.01
Num of Std Step Trials= 20
Max Error Tol= 0.3
Flow Tol Ratio= 0.001
Split Flow NTrial= 30
Split Flow Tol= 0.02
Split Flow Ratio= 0.02
Log Output Level= 0
Friction Slope Method= 1
Unsteady Friction Slope Method= 2
Unsteady Bridges Friction Slope Method= 1
Parabolic Critical Depth
Global Vel Dist=  1 , 1 , 1
Global Log Level= 0
CheckData=True
Encroach Param= -1, 0, 0, 0
BEGIN DESCRIPTION:
Multiple Run
END DESCRIPTION:

--- Catlett Creek.f01 (steady flow) ---

Flow Title=Multiple
Number of Profiles=7
Profile Names=10-year,25-year,50-year,1pct_min,100-year,1pct_plu,500-year
River Rch & RM= Catlett Creek,Reach-1,80251
     751    1049    1300     800    1596    3185    2413
River Rch & RM= Catlett Creek,Reach-1,76190
     802    1122    1392     858    1712    3415    2592
River Rch & RM= Catlett Creek,Reach-1,74326
     944    1331    1660    1027    2050    4089    3131
River Rch & RM= Catlett Creek,Reach-1,72333
    1109    1572    1968    1221    2437    4863    3747
River Rch & RM= Catlett Creek,Reach-1,68618
    1204    1714    2150    1337    2667    5321    4116
River Rch & RM= Catlett Creek,Reach-1,67942
    1647    2382    3021    1897    3785    7552    5959
River Rch & RM= Catlett Creek,Reach-1,65248
    1908    2766    3514    2208    4406    8792    6951
River Rch & RM= Catlett Creek,Reach-1,58164
    2121    3089    3936    2480    4949    9875    7850
River Rch & RM= Catlett Creek,Reach-1,53826
    3799    5668    7339    4693    9364   18683   15293
River Rch & RM= Catlett Creek,Reach-1,51757
    3980    5944    7702    4928    9833   19619   16076
River Rch & RM= Catlett Creek,Reach-1,48446
    3957    5894    7625    4869    9716   19385   15825
River Rch & RM= Catlett Creek,Reach-1,43562
    4210    6285    8142    5207   10389   20729   16969
River Rch & RM= Catlett Creek,Reach-1,43083
    4325    6458    8367    5351   10676   21302   17437
River Rch & RM= Catlett Creek,Reach-1,40256
    4460    6662    8634    5522   11019   21985   18002
River Rch & RM= Catlett Creek,Reach-1,38436
    4512    6741    8737    5588   11150   22247   18215
River Rch & RM= Catlett Creek,Reach-1,37087
    5493    8252   10738    6892   13751   27436   22617
River Rch & RM= Catlett Creek,Reach-1,33536
    5809    8740   11383    7312   14590   29110   24037
River Rch & RM= Catlett Creek,Reach-1,32677
    5697    8547   11109    7121   14208   28348   23308
River Rch & RM= Catlett Creek,Reach-1,29439
    5837    8756   11379    7293   14552   29034   23864
River Rch & RM= Catlett Creek,Reach-1,24945
    5931    8897   11564    7411   14787   29504   24248
River Rch & RM= Catlett Creek,Reach-1,19813
    6647    9993   13008    8347   16655   33231   27376
River Rch & RM= Catlett Creek,Reach-1,15677
    6655    9988   12986    8322   16604   33129   27220
River Rch & RM= Catlett Creek,Reach-1,10296
    7095   10656   13863    8888   17734   35383   29095
River Rch & RM= Catlett Creek,Reach-1,4456
    9006   13602   17765   11430   22806   45503   37670
Boundary for River Rch & Prof#=Catlett Creek,Reach-1,1
Up Type=0
Dn Type=1
Dn Known WS=751.7
Boundary for River Rch & Prof#=Catlett Creek,Reach-1,2
Up Type=0
Dn Type=1
Dn Known WS=752.88
Boundary for River Rch & Prof#=Catlett Creek,Reach-1,3
Up Type=0
Dn Type=1
Dn Known WS=753.68
Boundary for River Rch & Prof#=Catlett Creek,Reach-1,4
Up Type=0
Dn Type=1
Dn Known WS=752.38
Boundary for River Rch & Prof#=Catlett Creek,Reach-1,5
Up Type=0
Dn Type=1
Dn Known WS=754.38
Boundary for River Rch & Prof#=Catlett Creek,Reach-1,6
Up Type=0
Dn Type=1
Dn Known WS=756.75
Boundary for River Rch & Prof#=Catlett Creek,Reach-1,7
Up Type=0
Dn Type=1
Dn Known WS=756.02

--- Catlett Creek.g01 (geometry) ---

Geom Title=Existing Conditions

River Reach=Catlett Creek,Reach-1
Reach XY= 30
      2243179.00      7159660.00      2244411.69      7156926.27
      2252142.31      7151796.63      2253118.94      7149570.03
      2255209.37      7148930.15      2256684.03      7145407.69
      2257837.44      7144613.41      2261877.55      7145056.47
      2262676.29      7144165.40      2263655.71      7144183.67
      2263936.93      7142603.60      2265244.77      7141809.89
      2268344.11      7143009.73      2269923.31      7142461.87
      2271229.00      7143610.00      2273787.32      7141562.96
      2275594.16      7141160.36      2277570.53      7141262.58
      2277583.95      7142405.06      2278567.12      7142608.47
      2279285.03      7141961.61      2279923.59      7142204.82
      2282026.30      7138865.36      2285849.03      7138210.07
      2286804.01      7138810.43      2289323.14      7138407.94
      2290309.24      7138030.13      2290526.26      7137115.34
      2292845.77      7136443.57      2292729.00      7135360.00

Type RM Length L Ch R = 1,80251,591,591,591
BEGIN DESCRIPTION:
Catlett Creek 105.0
END DESCRIPTION:
XS GIS Cut Line= 3
      2243421.67      7159737.47      2243189.77      7159651.26
      2243007.09      7159585.39
#Sta/Elev= 30
  4740.7 1046.09  4786.2 1044.43  4826.3 1042.27  4834.1 1042.78  4850.2 1041.19
  4889.4 1039.49  4903.6 1039.13  4914.2 1039.56  4919.8 1038.93  4944.8 1038.77
  4950.1 1038.33  4967.6 1035.93  4980.5 1031.19  4983.8 1025.19  4984.1 1024.69
  4987.6 1024.69  4987.8 1025.19  4991.2 1025.19  4999.6 1030.50  5005.7 1033.39
  5020.8 1033.73  5036.4 1035.80  5052.7 1034.89  5061.8 1036.15  5067.1 1039.60
  5074.0 1041.06  5086.0 1041.81  5105.9 1042.68  5159.1 1046.69  5182.3 1047.67
#Mann=5,-1,0
  4740.7    0.05       0  4826.3    0.12       0  4983.8    0.07       0
  4987.8    0.12       0  5086.0    0.05       0
Bank Sta=4983.8,4987.8
Exp/Cntr=0.3,0.1

Type RM Length L Ch R = 1,79660,356,356,356
BEGIN DESCRIPTION:
Catlett Creek 104.0
END DESCRIPTION:
XS GIS Cut Line= 3
      2243757.71      7159455.73      2243328.74      7159340.04
      2243013.14      7159211.95
#Sta/Elev= 30
  4555.7 1046.53  4559.0 1045.74  4585.4 1045.67  4647.6 1043.05  4713.5 1042.52
  4720.1 1041.16  4740.8 1041.05  4761.5 1039.00  4778.7 1038.79  4822.9 1036.22
  4828.1 1036.79  4902.7 1034.97  4937.5 1035.16  4958.3 1033.78  4968.7 1032.63
  4977.4 1028.04  4982.6 1028.54  4995.3 1016.17  4995.5 1015.67  4999.3 1016.17
  5002.6 1016.17  5009.3 1018.43  5014.7 1017.61  5021.3 1022.45  5032.1 1027.06
  5044.1 1031.04  5048.1 1031.52  5086.1 1036.99  5092.3 1039.62  5340.6 1054.89
#Mann=5,-1,0
  4555.7    0.05       0  4778.7    0.12       0  4995.3    0.07       0
  4999.3    0.12       0  5048.1    0.05       0
Bank Sta=4995.3,4999.3
Exp/Cntr=0.3,0.1

Type RM Length L Ch R = 1,79304,348,348,348
BEGIN DESCRIPTION:
Catlett Creek 103.0
END DESCRIPTION:
XS GIS Cut Line= 3
      2243743.15      7159218.47      2243562.06      7159119.01
      2243273.53      7158962.19
#Sta/Elev= 30
  4793.4 1042.44  4840.1 1039.69  4905.5 1036.91  4955.6 1032.40  4965.2 1031.92
  4980.7 1024.56  4987.0 1020.78  4996.9 1011.08  4997.1 1010.58  5000.6 1010.58
  5000.9 1011.08  5004.2 1011.08  5014.9 1021.26  5025.0 1023.11  5030.6 1023.60
  5046.8 1023.05  5052.5 1023.80  5090.5 1024.51  5096.2 1026.50  5106.4 1027.58
  5112.4 1027.58  5118.1 1030.27  5128.5 1030.33  5134.2 1031.91  5140.1 1034.80
  5156.1 1035.54  5215.9 1040.60  5281.5 1044.05  5288.0 1045.24  5328.4 1047.87
#Mann=5,-1,0
  4793.4    0.05       0  4955.6    0.12       0  4996.9    0.07       0
  5000.9    0.12       0  5106.4    0.05       0
Bank Sta=4996.9,5000.9
Exp/Cntr=0.3,0.1

Type RM Length L Ch R = 1,78956,483,483,483
BEGIN DESCRIPTION:
Catlett Creek 102.0
END DESCRIPTION:
XS GIS Cut Line= 3
      2243985.90      7158951.59      2243700.10      7158869.72
      2243346.32      7158814.88
#Sta/Elev= 30
  4702.7 1045.08  4782.7 1039.95  4804.0 1040.58  4832.5 1037.49  4858.7 1035.62
  4876.7 1033.78  4886.7 1030.76  4897.1 1030.25  4944.2 1022.08  4969.9 1020.38
  4978.0 1018.89  4983.2 1019.29  4990.7 1015.26  4996.0 1007.90  4996.2 1007.40
  5000.0 1007.90  5003.1 1007.90  5021.3 1018.10  5028.6 1019.50  5033.7 1023.67
  5041.6 1026.39  5061.8 1028.04  5071.9 1027.47  5082.1 1024.87  5091.6 1019.88
  5098.0 1019.47  5102.3 1019.58  5132.7 1024.71  5159.7 1033.27  5358.0 1044.73
#Mann=5,-1,0
  4702.7    0.05       0  4858.7    0.12       0  4996.0    0.07       0
  5000.0    0.12       0  5098.0    0.05       0
Bank Sta=4996,5000
Exp/Cntr=0.3,0.1

Type RM Length L Ch R = 1,78473,521,521,521
BEGIN DESCRIPTION:
Catlett Creek 101.0
END DESCRIPTION:
XS GIS Cut Line= 3
      2244072.70      7158689.09      2243805.80      7158592.61
      2243496.94      7158477.26
#Sta/Elev= 30
  4716.2 1041.34  4814.6 1035.72  4844.2 1034.34  4858.4 1034.68  4874.8 1031.97
  4905.5 1030.22  4922.2 1030.71  4943.4 1028.51  4954.1 1025.51  4961.5 1021.59
  4966.8 1021.23  4986.0 1007.30  4990.1 1005.34  4990.4 1004.84  4994.1 1005.34
  5000.0 1005.58  5007.3 1009.69  5017.2 1013.21  5022.5 1012.70  5028.6 1015.13
  5047.5 1024.97  5052.8 1024.15  5060.6 1025.89  5071.3 1026.61  5083.1 1025.07
  5092.7 1025.42  5133.1 1029.61  5182.5 1032.35  5316.8 1039.71  5329.7 1039.17
#Mann=5,-1,0
  4716.2    0.05       0  4814.6    0.12       0  4990.1    0.07       0
  4994.1    0.12       0  5182.5    0.05       0
Bank Sta=4990.1,4994.1
Exp/Cntr=0.3,0.1

Type RM Length L Ch R = 1,77952,325,325,325
BEGIN DESCRIPTION:
Catlett Creek 100.0
END DESCRIPTION:
XS GIS Cut Line= 3
      2244143.39      7158281.00      2243900.38      7158246.87
      2243605.97      7158214.34
#Sta/Elev= 30
  4754.6 1035.32  4789.3 1034.36  4811.8 1032.49  4849.9 1030.63  4880.2 1027.47
  4920.6 1025.57  4930.7 1024.20  4938.7 1019.52  4943.7 1020.44  4950.9 1016.47
  4971.1 1011.14  4981.2 1009.50  4991.3 1003.97  4996.2  998.18  4996.4  997.68
  5000.2  998.18  5003.2  998.18  5011.4 1004.33  5016.8 1017.43  5021.8 1013.04
  5031.6 1017.93  5041.6 1018.17  5061.8 1024.85  5102.0 1027.58  5107.6 1028.80
  5192.5 1033.69  5198.4 1034.62  5212.7 1034.76  5263.0 1038.55  5296.2 1039.60
#Mann=4,-1,0
  4754.6    0.05       0  4811.8    0.12       0  4996.2    0.07       0
  5000.2    0.12       0
Bank Sta=4996.2,5000.2
Exp/Cntr=0.3,0.1

Type RM Length L Ch R = 1,77627,520,520,520
BEGIN DESCRIPTION:
Catlett Creek 99.0
END DESCRIPTION:
XS GIS Cut Line= 3
      2244167.67      7158069.12      2243897.75      7157962.53
      2243733.11      7157905.32
#Sta/Elev= 30
  4709.8 1030.82  4732.5 1029.40  4752.5 1028.70  4825.6 1023.18  4837.4 1023.60
  4855.3 1022.80  4869.6 1020.74  4879.7 1020.28  4885.1 1018.82  4891.1 1020.25
  4901.9 1016.83  4914.8 1013.97  4923.4 1009.62  4933.8 1007.93  4939.2 1006.12
  4944.9 1005.47  4963.5 1006.01  4977.2 1004.69  4993.3  996.97  4994.6  994.26
  4994.9  993.76  4998.6  994.26  5000.0  994.26  5009.3  998.60  5018.7 1007.25
  5024.0 1008.37  5041.0 1020.61  5049.9 1025.11  5157.5 1029.11  5174.3 1030.34
#Mann=4,-1,0
  4709.8    0.05       0  4732.5    0.12       0  4994.6    0.07       0
  4998.6    0.12       0
Bank Sta=4994.6,4998.6
Exp/Cntr=0.3,0.1

Type RM Length L Ch R = 1,77107,249,249,249
BEGIN DESCRIPTION:
Catlett Creek 98.0
END DESCRIPTION:
XS GIS Cut Line= 3
      2244269.01      7157823.62      2243995.64      7157603.62
      2243762.72      7157401.79
#Sta/Elev= 30
  4649.1 1027.58  4708.8 1023.24  4758.4 1021.20  4764.8 1021.94  4818.9 1018.74
  4929.5 1018.08  4943.9 1016.53  4950.4 1014.65  4957.2 1008.52  4979.1  999.27
  4985.6  991.21  4991.5  986.06  4991.8  985.56  4995.5  986.06  5014.3  990.90
  5021.9  994.80  5035.3 1007.45  5042.8 1007.20  5049.4 1009.81  5057.0 1009.31
  5063.7 1012.40  5077.9 1012.85  5085.5 1016.14  5092.2 1015.84  5099.8 1017.84
  5106.4 1017.24  5114.0 1018.83  5134.9 1020.14  5171.3 1021.14  5308.2 1027.64
#Mann=5,-1,0
  4649.1    0.05       0  4818.9    0.12       0  4991.5    0.07       0
  4995.5    0.12       0  5171.3    0.05       0
Bank Sta=4991.5,4995.5
Exp/Cntr=0.3,0.1

Type RM Length L Ch R = 1,76858,367,367,367
BEGIN DESCRIPTION:
Mapping XS 162fba7a
END DESCRIPTION:
XS GIS Cut Line= 3
      2244298.88      7157624.86      2244155.24      7157422.79
      2243895.83      7157244.48
#Sta/Elev= 30
  4720.0 1020.73  4813.9 1016.99  4887.7 1016.10  4910.0 1012.06  4917.2 1007.80
  4923.3 1014.55  4932.0 1016.00  4938.1 1006.45  4946.7 1004.63  4952.9  992.71
  4959.1  990.13  4966.6  990.00  4973.5  982.16  4973.7  981.66  4977.5  982.16
  4981.6  986.95  4996.5  988.03  5002.6  984.31  5011.4  987.72  5017.5  986.72
  5038.4  999.68  5047.3 1012.41  5053.3 1013.95  5089.2 1016.15  5104.1 1015.49
  5119.0 1017.27  5125.0 1015.35  5139.9 1019.14  5151.0 1018.86  5282.7 1022.94
#Mann=5,-1,0
  4720.0    0.05       0  4813.9    0.12       0  4973.5    0.07       0
  4977.5    0.12       0  5151.0    0.05       0
Bank Sta=4973.5,4977.5
Exp/Cntr=0.3,0.1

Type RM Length L Ch R = 1,76491,301,301,301
BEGIN DESCRIPTION:
Catlett Creek 96.0
END DESCRIPTION:
XS GIS Cut Line= 3
      2244639.27      7157482.95      2244425.94      7157251.72
      2244002.66      7156948.81
#Sta/Elev= 30
  4685.4 1027.09  4793.9 1022.04  4906.0 1018.93  4935.1 1018.05  4949.3 1016.19
  4956.7 1009.34  4963.5 1001.17  4977.7  988.51  4985.0  984.72  4991.8  983.63
  4995.8  979.69  4996.0  979.19  4999.8  979.69  5007.0  981.07  5013.1  988.49
  5027.9  996.81  5042.6 1009.03  5048.7 1008.19  5057.3 1011.79  5063.5 1009.72
  5078.2 1013.23  5099.1 1011.29  5156.1 1011.73  5170.4 1010.35  5179.0 1006.45
  5214.6 1009.04  5235.5 1013.25  5297.6 1016.82  5401.3 1019.86  5520.5 1026.02
#Mann=5,-1,0
  4685.4    0.05       0  4906.0    0.12       0  4995.8    0.07       0
  4999.8    0.12       0  5297.6    0.05       0
Bank Sta=4995.8,4999.8
Exp/Cntr=0.3,0.1

Type RM Length L Ch R = 1,76190,185,185,185
BEGIN DESCRIPTION:
Mapping XS 7ad3d1b1
END DESCRIPTION:
XS GIS Cut Line= 3
      2244648.66      7157195.01      2244510.51      7157027.60
      2244103.06      7156841.00
#Sta/Elev= 30
  4639.5 1018.19  4657.5 1017.03  4678.3 1017.31  4692.7 1015.24  4707.2 1015.00
  4756.5 1012.94  4777.3 1013.48  4806.0 1011.24  4859.7 1010.78  4863.3 1007.48
  4880.2 1006.42  4886.3 1004.13  4891.8  999.85  4902.2  996.84  4924.2  993.18
  4937.8  989.25  4955.3  982.73  4960.8  982.71  4968.2  978.14  4976.3  978.00
  4976.5  977.50  4980.3  978.00  4983.8  978.92  4986.8  985.81  4990.2  993.61
  5001.2 1005.73  5006.8 1009.91  5023.2 1012.44  5081.3 1014.11  5304.7 1025.16
#Mann=5,-1,0
  4639.5    0.05       0  4707.2    0.12       0  4976.3   0.033       0
  4980.3    0.12       0  4986.8    0.05       0
Bank Sta=4976.3,4980.3
Exp/Cntr=0.3,0.1

Type RM Length L Ch R = 1,76005,521,521,521
BEGIN DESCRIPTION:
Catlett Creek 95.0
END DESCRIPTION:
XS GIS Cut Line= 3
      2244760.45      7157228.40      2244538.98      7156910.06
      2244262.89      7156581.31
#Sta/Elev= 30
  4612.2 1022.15  4670.5 1020.79  4706.3 1017.81  4802.7 1013.08  4906.2 1010.32
  4914.8 1006.96  4935.9  994.28  4950.7  987.84  4971.7  980.56  4990.5  977.23
  4990.8  976.73  4994.6  977.23  4997.0  980.25  5003.3  980.25  5007.2  985.25
  5009.9  986.43  5013.7  988.09  5035.8 1003.64  5042.3 1009.41  5056.6 1011.50
  5085.2 1011.24  5156.7 1013.70  5177.6 1013.11  5184.1 1014.12  5198.4 1014.17
  5204.7 1012.53  5234.8 1015.52  5376.6 1022.77  5397.4 1022.97  5429.3 1026.56
#Mann=6,-1,0
  4612.2    0.05       0  4802.7    0.12       0  4990.5    0.07       0
  4994.6    0.12       0  5009.9    0.05       0  5204.7    0.12       0
Bank Sta=4990.5,4994.6
Exp/Cntr=0.3,0.1

Type RM Length L Ch R = 1,75484,282,282,282
BEGIN DESCRIPTION:
Catlett Creek 94.0
END DESCRIPTION:
XS GIS Cut Line= 3
      2245082.00      7156999.89      2244937.02      7156703.66
      2244776.04      7156489.52
#Sta/Elev= 30
  4670.2 1018.05  4853.8 1011.37  4895.7 1010.32  4903.9 1008.92  4926.1 1000.96
  4935.2  999.28  4940.7  994.69  4948.4  993.48  4957.7  997.67  4963.2  991.93
  4970.7  992.00  4980.2  986.01  4985.8  979.51  4997.2  973.15  4997.5  972.65
  5001.3  973.15  5002.5  973.15  5016.3  981.83  5029.6  992.27  5037.1  996.07
  5043.3  996.99  5051.7 1000.78  5057.9 1002.21  5066.2 1006.22  5079.6 1007.16
  5207.9 1007.56  5222.4 1009.04  5229.8 1008.36  5251.6 1010.40  5267.9 1010.47
#Mann=4,-1,0
  4670.2    0.05       0  4853.8    0.12       0  4997.2    0.07       0
  5001.3    0.12       0
Bank Sta=4997.2,5001.3
Exp/Cntr=0.3,0.1

Type RM Length L Ch R = 1,75202,266,266,266
BEGIN DESCRIPTION:
Catlett Creek 93.0
END DESCRIPTION:
XS GIS Cut Line= 3
      2245309.26      7156713.26      2245173.07      7156568.44
      2245004.41      7156398.69
#Sta/Elev= 30
  4801.2 1013.21  4824.9 1012.85  4839.0 1011.92  4846.3 1010.48  4860.5 1010.68
  4881.5 1008.76  4915.6 1007.68  4924.0 1006.49  4945.0 1005.81  4952.3 1002.88
  4966.5  993.98  4973.4  993.70  4980.7  988.51  4987.5  980.03  4992.7  970.83
  4993.1  970.33  4996.9  970.83  4999.3  972.90  5030.1  978.93  5037.1  982.77
  5051.3  994.22  5065.4 1000.69  5079.6 1003.86  5093.7 1003.10  5136.1 1004.98
  5143.2 1004.07  5192.7 1004.97  5206.9 1005.83  5213.9 1007.35  5239.3 1007.10
#Mann=4,-1,0
  4801.2    0.05       0  4915.6    0.12       0  4992.7    0.07       0
  4996.9    0.12       0
Bank Sta=4992.7,4996.9
Exp/Cntr=0.3,0.1

Type RM Length L Ch R = 1,74936,425,425,425
BEGIN DESCRIPTION:
Catlett Creek 92.0
END DESCRIPTION:
XS GIS Cut Line= 3
      2245557.19      7156591.74      2245377.85      7156410.89
      2245194.71      7156170.25
#Sta/Elev= 30
  4745.3 1003.57  4858.4 1003.43  4895.2 1003.94  4907.9 1003.42  4915.0 1004.07
  4929.1 1000.59  4936.2 1000.76  4950.3  996.67  4957.4  989.71  4971.5  978.89
  4985.7  973.20  4992.7  973.40  4995.0  970.33  4995.4  969.83  4998.9  969.83
  4999.2  970.33  5006.9  971.10  5013.7  979.05  5021.4  985.67  5027.7  988.48
  5036.0  995.00  5042.2  996.45  5050.5  999.80  5056.8 1001.07  5100.4 1003.21
  5171.1 1004.09  5227.3 1007.28  5250.1 1007.49  5291.7 1009.43  5302.4 1009.37
#Mann=4,-1,0
  4745.3    0.05       0  4895.2    0.12       0  4995.0    0.07       0
  4999.2    0.12       0
Bank Sta=4995,4999.2
Exp/Cntr=0.3,0.1

Type RM Length L Ch R = 1,74511,185,185,185
BEGIN DESCRIPTION:
Catlett Creek 91.5
END DESCRIPTION:
XS GIS Cut Line= 3
      2245641.92      7156472.27      2245722.96      7156218.18
      2245423.93      7155905.71
#Sta/Elev= 30
  4733.3 1001.66  4849.0 1000.15  4882.6 1000.36  4893.1  995.36  4901.5  992.99
  4906.8  995.87  4914.1  991.32  4933.7  983.53  4939.0  984.41  4965.9  975.63
  4971.2  977.83  4996.4  968.68  5006.5  968.61  5006.9  968.11  5010.8  968.61
  5022.8  978.51  5051.1  981.25  5058.1  984.90  5065.3  984.43  5072.2  988.99
  5086.4  992.28  5093.6  992.26  5100.5  990.28  5107.8  995.02  5114.7  993.50
  5121.9  995.81  5128.8  995.16  5143.0  997.68  5227.9  999.87  5432.5 1010.14
#Mann=4,-1,0
  4733.3    0.05       0  4849.0    0.12       0  5006.5    0.07       0
  5010.8    0.12       0
Bank Sta=5006.5,5010.8
Exp/Cntr=0.3,0.1

Type RM Length L Ch R = 1,74326,425,425,425
BEGIN DESCRIPTION:
Catlett Creek 91.0
END DESCRIPTION:
XS GIS Cut Line= 3
      2246063.40      7156238.85      2245827.12      7156098.75
      2245606.02      7155874.24
#Sta/Elev= 30
  4725.3  995.41  4787.2  993.92  4800.2  992.27  4808.6  992.81  4814.4  990.99
  4858.3  989.37  4881.6  980.70  4888.5  984.31  4894.4  981.06  4904.2  983.40
  4910.0  979.42  4925.6  980.59  4931.4  979.27  4952.8  979.07  4962.6  970.30
  4968.4  976.13  4974.6  969.64  4984.1  971.12  4987.5  967.05  4988.0  966.55
  4992.3  967.05  5002.2  967.64  5026.1  979.00  5033.1  980.06  5040.3  984.09
  5047.3  985.35  5061.4  994.11  5075.6  995.93  5167.4  998.60  5315.1 1008.49
#Mann=3,-1,0
  4725.3    0.12       0  4987.5    0.07       0  4992.3    0.12       0
Bank Sta=4987.5,4992.3
Exp/Cntr=0.3,0.1

Type RM Length L Ch R = 1,73901,291,291,291
BEGIN DESCRIPTION:
Mapping XS 660be2f5
END DESCRIPTION:
XS GIS Cut Line= 2
      2246073.28      7156223.81      2246071.47      7155759.72
#Sta/Elev= 30
  4735.0  994.79  4768.8  993.22  4778.8  992.15  4788.8  987.49  4798.8  986.93
  4828.8  991.87  4848.8  991.49  4868.8  992.01  4878.8  989.92  4898.8  990.01
  4908.8  986.38  4918.8  985.23  4948.8  972.58  4958.8  969.06  4968.8  967.60
  4978.8  967.47  4988.8  966.37  4996.4  963.49  4997.0  962.99  5001.2  963.49
  5008.8  966.09  5018.8  971.39  5028.8  974.05  5038.8  978.57  5048.8  979.76
  5058.8  984.73  5078.8  987.57  5088.8  988.04  5118.8  998.30  5199.1 1001.64
#Mann=3,-1,0
  4735.0    0.12       0  4996.4    0.07       0  5001.2    0.12       0
Bank Sta=4996.4,5001.2
Exp/Cntr=0.3,0.1

Type RM Length L Ch R = 1,73610,320,320,320
BEGIN DESCRIPTION:
Catlett Creek 90.0
END DESCRIPTION:
XS GIS Cut Line= 3
      2246305.09      7156357.36      2246290.19      7156109.50
      2246198.76      7155719.37
#Sta/Elev= 30
  4751.7 1004.05  4859.2  999.15  4908.3  997.99  4929.4  994.90  4935.4  989.42
  4940.5  989.79  4949.4  985.32  4979.5  975.37  4989.5  969.94  4994.8  963.52
  4995.4  963.02  4999.7  963.52  5009.8  963.67  5020.0  968.20  5031.3  970.49
  5040.6  969.79  5050.8  972.25  5061.1  976.59  5068.6  976.99  5073.7  979.80
  5111.1  986.76  5116.2  989.23  5143.3  988.74  5158.6  991.04  5163.8  990.02
  5201.1  989.94  5206.2  990.97  5225.5  990.01  5307.6  992.63  5400.7  998.65
#Mann=4,-1,0
  4751.7    0.05       0  4908.3    0.12       0  4994.8    0.07       0
  4999.7    0.12       0
Bank Sta=4994.8,4999.7
Exp/Cntr=0.3,0.1

Type RM Length L Ch R = 1,73290,354,354,354
BEGIN DESCRIPTION:
Catlett Creek 89.0
END DESCRIPTION:
XS GIS Cut Line= 3
      2246636.06      7156036.20      2246476.92      7155904.29
      2246233.18      7155706.97
#Sta/Elev= 30
  4793.3  996.52  4902.4  989.57  4931.0  980.40  4937.5  980.32  4945.3  976.89
  4951.9  975.34  4958.4  971.18  4972.7  973.22  4980.5  967.95  4987.0  972.77
  4994.8  964.65  4996.9  960.81  4997.6  960.31  5001.9  960.81  5023.1  966.17
  5030.1  969.50  5036.5  970.24  5044.5  973.66  5050.9  974.21  5058.8  977.96
  5065.3  979.34  5079.6  985.78  5094.0  989.32  5108.4  989.86  5129.2  988.63
  5172.4  991.93  5193.2  991.44  5250.7  993.56  5257.1  994.76  5313.6  998.28
#Mann=3,-1,0
  4793.3    0.12       0  4996.9    0.07       0  5001.9    0.12       0
Bank Sta=4996.9,5001.9
Exp/Cntr=0.3,0.1

Type RM Length L Ch R = 1,72936,393,393,393
BEGIN DESCRIPTION:
Catlett Creek 88.0
END DESCRIPTION:
XS GIS Cut Line= 3
      2246804.00      7155735.00      2246528.63      7155566.38
      2246237.84      7155428.56
#Sta/Elev= 30
  4677.1  993.86  4741.6  988.28  4793.2  985.97  4829.9  985.93  4858.9  988.24
  4903.4  985.18  4917.5  985.74  4924.7  983.99  4930.6  984.23  4940.1  979.97
  4946.0  979.97  4961.4  969.94  4967.3  970.07  4976.1  963.79  4982.7  962.13
  5000.0  962.86  5001.7  961.79  5002.3  961.29  5006.7  961.79  5010.7  968.75
  5021.4  973.47  5026.9  974.46  5032.8  979.63  5043.9  986.79  5049.7  989.74
  5055.2  990.73  5140.6  998.61  5276.2 1006.67  5310.9 1010.88  5321.8 1010.92
#Mann=3,-1,0
  4677.1    0.12       0  5001.7    0.07       0  5006.7    0.12       0
Bank Sta=5001.7,5006.7
Exp/Cntr=0.3,0.1

Type RM Length L Ch R = 1,72543,210,210,210
BEGIN DESCRIPTION:
Catlett Creek 87.5
END DESCRIPTION:
XS GIS Cut Line= 3
      2247039.65      7155531.60      2246815.61      7155373.68
      2246404.96      7155235.42
#Sta/Elev= 30
  4725.9  986.78  4791.7  985.86  4800.1  984.26  4877.9  979.10  4892.7  980.21
  4928.4  978.63  4949.3  979.53  4958.0  975.70  4964.1  975.53  4978.9  964.90
  4985.0  966.13  4993.7  956.80  4996.4  956.77  4997.0  956.27  5001.4  956.77
  5007.0  957.86  5025.0  966.58  5030.3  966.08  5038.6  969.79  5049.2  972.75
  5061.8  975.89  5080.8  978.73  5088.0  982.49  5133.6  988.04  5151.0  989.94
  5175.8  990.86  5260.2  999.19  5270.8  999.06  5376.7 1005.95  5433.3 1007.78
#Mann=3,-1,0
  4725.9    0.12       0  4996.4    0.07       0  5001.4    0.12       0
Bank Sta=4996.4,5001.4
Exp/Cntr=0.3,0.1

Type RM Length L Ch R = 1,72333,439,439,439
BEGIN DESCRIPTION:
Catlett Creek 87.0
END DESCRIPTION:
XS GIS Cut Line= 3
      2247044.04      7155522.82      2246952.19      7155250.91
      2246982.90      7155005.53
#Sta/Elev= 30
  4713.0  987.02  4800.4  983.61  4821.5  980.08  4837.7  978.96  4843.0  980.26
  4853.2  980.40  4863.7  978.92  4869.2  976.48  4884.9  975.50  4906.0  977.51
  4948.2  978.27  4958.3  976.08  4963.6  976.26  4969.3  973.66  4989.7  960.18
  4995.0  959.76  4995.2  954.60  4995.9  954.10  5000.4  954.60  5003.0  954.60
  5010.3  961.24  5015.3  960.86  5021.1  961.98  5031.2  966.84  5041.2  974.94
  5081.5  979.21  5101.7  984.06  5121.9  985.17  5176.5  984.80  5247.3  986.70
#Mann=3,-1,0
  4713.0    0.12       0  4995.2    0.07       0  5000.4    0.12       0
Bank Sta=4995.2,5000.4
Exp/Cntr=0.3,0.1

Type RM Length L Ch R = 1,71894,388,388,388
BEGIN DESCRIPTION:
Catlett Creek 86.0
END DESCRIPTION:
XS GIS Cut Line= 3
      2247346.10      7155356.17      2247325.39      7155208.52
      2247030.10      7154962.41
#Sta/Elev= 30
  4850.9  980.09  4935.4  976.63  4940.5  969.08  4958.1  959.04  4968.2  954.75
  4985.8  953.24  4986.5  952.74  4991.0  953.24  5000.0  953.59  5003.7  957.53
  5032.3  965.00  5060.4  963.85  5067.4  968.70  5073.9  968.24  5081.8  973.99
  5088.3  973.27  5096.1  976.05  5131.2  975.10  5145.5  977.82  5180.7  974.01
  5202.8  975.84  5223.6  973.95  5230.1  977.27  5238.0  975.21  5258.8  980.20
  5266.6  977.30  5273.1  979.40  5280.9  977.62  5308.2  984.35  5384.4  985.25
#Mann=3,-1,0
  4850.9    0.12       0  4985.8    0.07       0  4991.0    0.12       0
Bank Sta=4985.8,4991
Exp/Cntr=0.3,0.1

Type RM Length L Ch R = 1,71506,309,309,309
BEGIN DESCRIPTION:
Catlett Creek 85.0
END DESCRIPTION:
XS GIS Cut Line= 3
      2247679.69      7155472.36      2247503.88      7154909.48
      2247267.35      7154645.96
#Sta/Elev= 30
  4410.3  990.00  4486.1  985.82  4493.8  984.08  4629.1  976.53  4829.2  972.76
  4861.7  969.11  4867.0  970.66  4873.7  968.14  4894.2  966.62  4899.4  971.14
  4905.2  970.95  4931.9  964.06  4937.2  965.67  4969.7  961.98  4989.0  956.45
  4996.9  952.62  4997.0  950.81  4997.8  950.31  5002.6  950.81  5024.6  961.76
  5045.5  963.89  5053.0  966.94  5059.7  965.75  5073.9  973.71  5080.7  973.73
  5102.3  979.18  5180.1  981.55  5222.7  985.14  5288.9  987.91  5354.1  992.19
#Mann=5,-1,0
  4410.3    0.05       0  4493.8    0.12       0  4997.0    0.07       0
  5002.6    0.12       0  5288.9    0.05       0
Bank Sta=4997,5002.6
Exp/Cntr=0.3,0.1

Type RM Length L Ch R = 1,71197,293,293,293
BEGIN DESCRIPTION:
Mapping XS 752419cf
END DESCRIPTION:
XS GIS Cut Line= 3
      2247809.14      7155255.34      2247814.34      7154992.21
      2247574.96      7154429.16
#Sta/Elev= 30
  4652.2  973.52  4797.6  971.37  4817.6  969.99  4937.9  969.79  4950.4  967.78
  4961.2  963.07  4967.0  958.89  4972.5  952.20  4983.0  949.68  4987.9  949.66
  4988.7  949.16  4993.5  949.66  4996.1  954.61  5014.3  956.55  5026.4  963.63
  5037.3  966.82  5043.4  966.06  5048.8  967.86  5059.0  967.33  5090.7  971.62
  5119.8  971.91  5125.2  973.61  5143.4  973.28  5148.8  975.42  5211.2  979.08
  5232.9  979.14  5402.2  990.41  5430.7  993.06  5472.0  994.01  5527.2  997.72
#Mann=4,-1,0
  4652.2    0.12       0  4987.9    0.07       0  4993.5    0.12       0
  5402.2    0.05       0
Bank Sta=4987.9,4993.5
Exp/Cntr=0.3,0.1

Type RM Length L Ch R = 1,70904,272,272,272
BEGIN DESCRIPTION:
Mapping XS 94553f19
END DESCRIPTION:
XS GIS Cut Line= 2
      2248133.92      7155029.61      2247790.68      7154414.38
#Sta/Elev= 30
  4633.8  978.45  4733.5  974.48  4760.9  971.98  4836.3  967.96  4858.0  967.22
  4885.5  967.93  4895.7  967.45  4917.4  962.88  4923.2  959.95  4944.9  958.15
  4979.7  957.28  4980.6  956.78  4985.5  957.28  4988.3  958.37  5004.3  960.95
  5011.2  966.21  5020.3  970.53  5026.0  969.81  5034.1  971.54  5063.7  974.63
  5160.1  980.66  5166.6  981.92  5210.0  985.53  5217.4  986.91  5263.2  989.66
  5269.4  990.95  5288.8  991.66  5297.5  992.61  5334.5  993.72  5338.3  994.56
#Mann=4,-1,0
  4633.8    0.12       0  4979.7    0.07       0  4985.5    0.12       0
  5288.8    0.05       0
Bank Sta=4979.7,4985.5
Exp/Cntr=0.3,0.1

Type RM Length L Ch R = 1,70632,507,507,507
BEGIN DESCRIPTION:
Catlett Creek 83.0
END DESCRIPTION:
XS GIS Cut Line= 3
      2248297.93      7154898.26      2248210.91      7154660.05
      2248050.52      7154377.39
#Sta/Elev= 30
  4746.4  978.57  4840.2  972.38  4870.7  969.16  4876.0  969.78  4884.3  968.15
  4901.2  964.51  4906.6  964.97  4914.9  960.84  4925.5  959.22  4957.0  956.02
  4962.3  956.56  4978.8  949.23  4987.5  949.31  4992.9  951.87  4997.4  949.50
  5009.9  950.23  5012.8  948.42  5013.7  947.92  5018.6  948.42  5023.1  950.87
  5031.5  958.09  5037.3  956.15  5046.1  963.50  5069.0  963.57  5096.4  966.44
  5126.5  967.56  5171.4  970.69  5214.7  975.17  5258.0  978.18  5325.0  986.07
#Mann=4,-1,0
  4746.4    0.05       0  4884.3    0.12       0  5012.8    0.07       0
  5018.6    0.12       0
Bank Sta=5012.8,5018.6
Exp/Cntr=0.3,0.1

Type RM Length L Ch R = 1,70125,386,386,386
BEGIN DESCRIPTION:
Catlett Creek 82.0
END DESCRIPTION:
XS GIS Cut Line= 3
      2248673.52      7154701.90      2248559.02      7154460.04
      2248344.77      7154129.97
#Sta/Elev= 30
  4732.4  974.46  4822.7  967.41  4866.6  960.55  4878.3  957.07  4889.4  959.36
  4894.9  961.80  4940.4  957.86  4968.7  957.48  4977.9  954.45  4985.9  947.16
  4991.4  948.27  4994.3  946.24  4995.3  945.74  5000.2  946.24  5003.0  946.24
  5007.6  952.19  5022.8  956.28  5035.8  956.97  5065.0  962.22  5101.2  964.48
  5110.7  966.31  5131.2  968.79  5152.6  969.14  5166.9  972.32  5188.9  972.48
  5215.9  975.23  5267.3  976.83  5297.6  979.97  5310.0  979.83  5393.5  985.88
#Mann=5,-1,0
  4732.4    0.05       0  4822.7    0.12       0  4994.3    0.07       0
  5000.2    0.12       0  5110.7    0.05       0
Bank Sta=4994.3,5000.2
Exp/Cntr=0.3,0.1

Type RM Length L Ch R = 1,69739,300,300,300
BEGIN DESCRIPTION:
Catlett Creek 81.0
END DESCRIPTION:
XS GIS Cut Line= 3
      2249016.04      7154596.20      2248888.81      7154399.57
      2248578.99      7153959.98
#Sta/Elev= 30
  4765.8  973.56  4768.4  972.78  4825.8  971.81  4840.9  969.82  4877.2  968.31
  4911.2  964.69  4955.7  960.68  4963.8  956.50  4970.9  956.42  4976.8  953.14
  4986.0  952.53  4992.0  944.36  5004.0  944.28  5005.0  943.78  5009.9  944.28
  5021.8  945.53  5027.9  948.72  5036.2  955.23  5042.7  956.99  5048.8  955.77
  5083.3  955.64  5121.8  956.88  5236.0  957.04  5250.8  957.36  5265.6  959.25
  5301.3  959.92  5366.5  965.77  5402.3  970.15  5501.1  984.89  5537.8  988.56
#Mann=5,-1,0
  4765.8    0.05       0  4911.2    0.12       0  5004.0    0.07       0
  5009.9    0.12       0  5083.3    0.05       0
Bank Sta=5004,5009.9
Exp/Cntr=0.3,0.1

Type RM Length L Ch R = 1,69439,368,368,368
BEGIN DESCRIPTION:
Mapping XS 650d7f36
END DESCRIPTION:
XS GIS Cut Line= 2
      2249218.32      7154408.82      2248820.11      7153803.92
#Sta/Elev= 30
  4762.1  972.20  4789.4  970.63  4825.5  965.39  4879.8  960.94  4891.8  961.35
  4904.4  959.13  4934.0  957.46  4940.3  955.32  4949.0  955.30  4955.0  954.10
  4985.2  952.85  4991.2  953.55  5000.1  950.71  5003.3  942.98  5004.2  942.48
  5009.2  942.98  5012.2  944.42  5027.3  944.35  5036.0  948.37  5042.4  953.96
  5048.4  955.18  5097.4  954.52  5143.8  955.41  5208.0  955.03  5259.3  956.43
  5280.3  958.34  5310.5  958.89  5346.6  961.00  5373.7  963.64  5486.3  970.98
#Mann=5,-1,0
  4762.1    0.05       0  4879.8    0.12       0  5003.3    0.07       0
  5009.2    0.12       0  5097.4    0.05       0
Bank Sta=5003.3,5009.2
Exp/Cntr=0.3,0.1

Type RM Length L Ch R = 1,69071,453,453,453
BEGIN DESCRIPTION:
Mapping XS 6643a5a3
END DESCRIPTION:
XS GIS Cut Line= 2
      2249481.05      7154293.34      2249030.41      7153684.22
#Sta/Elev= 30
  4579.7  967.99  4584.9  967.99  4590.8  967.02  4597.0  967.74  4605.4  967.10
  4611.7  967.80  4670.2  964.15  4726.5  962.41  4733.1  960.75  4755.7  958.64
  4808.9  955.73  4855.9  953.97  4897.6  953.60  4969.5  951.40  4977.0  948.60
  4983.2  948.62  4991.6  943.62  4997.8  941.89  5003.2  941.78  5004.2  941.28
  5009.2  941.78  5019.9  948.93  5027.1  953.41  5033.3  955.08  5112.6  955.56
  5127.3  957.08  5133.5  956.59  5192.0  958.54  5248.3  958.98  5337.4  961.37
#Mann=5,-1,0
  4579.7    0.05       0  4808.9    0.12       0  5003.2    0.07       0
  5009.2    0.12       0  5019.9    0.05       0
Bank Sta=5003.2,5009.2
Exp/Cntr=0.3,0.1

Type RM Length L Ch R = 1,68618,140,140,140
BEGIN DESCRIPTION:
Catlett Creek 78.0
END DESCRIPTION:
XS GIS Cut Line= 3
      2249719.88      7154178.35      2249628.88      7153809.72
      2249406.26      7153356.88
#Sta/Elev= 30
  4620.3  969.17  4659.8  964.11  4762.8  955.64  4793.7  955.48  4824.6  952.94
  4857.1  955.05  4876.1  952.01  4887.0  953.04  4893.4  951.47  4907.0  950.93
  4948.2  951.81  4976.3  949.16  4981.5  949.99  4989.4  946.09  4994.0  939.88
  4995.1  939.38  5000.5  939.88  5002.6  939.88  5008.2  945.69  5013.7  949.43
  5022.0  950.62  5133.0  952.74  5261.0  955.94  5289.4  956.00  5300.4  954.34
  5311.7  955.97  5373.4  957.81  5434.3  957.64  5440.8  956.68  5504.6  960.54
#Mann=5,-1,0
  4620.3    0.05       0  4887.0    0.12       0  4994.0    0.07       0
  5000.5    0.12       0  5133.0    0.05       0
#XS Ineff=2,0
       0                 5199.90    0.00  961.85
Permanent Ineff=
       F       F
Bank Sta=4994,5000.5
Exp/Cntr=0.3,0.1

Type RM Length L Ch R = 1,68478,223,223,223
BEGIN DESCRIPTION:
Mapping XS a9194583
END DESCRIPTION:
XS GIS Cut Line= 2
      2249855.71      7154023.08      2249494.79      7153113.79
#Sta/Elev= 30
  4738.9  959.10  4775.3  958.22  4806.8  954.92  4839.0  953.75  4883.3  950.11
  4907.6  950.53  4927.6  949.26  4956.2  948.88  4978.9  950.03  4991.3  948.73
  5000.4  942.15  5007.0  938.97  5008.0  938.47  5013.5  938.97  5015.6  939.70
  5022.0  945.13  5032.7  949.62  5069.1  949.08  5099.3  951.03  5140.3  950.64
  5334.0  953.63  5363.9  952.38  5417.9  954.61  5441.5  954.15  5453.0  955.81
  5484.6  956.24  5538.4  960.13  5602.9  962.18  5693.3  969.50  5717.2  972.39
#Mann=5,-1,0
  4738.9    0.05       0  4927.6    0.12       0  5007.0    0.07       0
  5013.5    0.12       0  5069.1    0.05       0
#XS Ineff=2,0
       0                 5200.00    0.00  960.89
Permanent Ineff=
       F       F
Bank Sta=5007,5013.5
Exp/Cntr=0.3,0.1

Type RM Length L Ch R = 1,68255,313,313,313
BEGIN DESCRIPTION:
Mapping XS daae628d
END DESCRIPTION:
XS GIS Cut Line= 3
      2249935.66      7153861.06      2249914.15      7153659.96
      2249597.98      7152983.44
#Sta/Elev= 30
  4797.2  956.67  4813.1  956.33  4878.7  950.10  4898.8  950.46  4922.9  948.05
  4969.2  946.51  4979.3  944.34  4986.1  939.10  4987.1  938.60  4992.6  939.10
  4996.9  941.12  4999.4  941.12  5002.4  939.45  5010.4  943.94  5019.7  947.70
  5027.4  948.75  5054.6  948.14  5076.7  949.26  5099.3  948.70  5213.5  950.78
  5253.3  949.51  5259.2  950.53  5310.4  952.25  5333.3  952.47  5341.6  951.52
  5407.8  954.78  5440.9  954.79  5463.0  956.86  5529.2  960.49  5746.2  971.14
#Mann=5,-1,0
  4797.2    0.05       0  4922.9    0.12       0  4986.1    0.07       0
  4992.6    0.12       0  5027.4    0.05       0
#XS Ineff=2,0
       0                 5182.50    0.00  959.25
Permanent Ineff=
       F       F
Bank Sta=4986.1,4992.6
Exp/Cntr=0.3,0.1

Type RM Length L Ch R = 1,67942,374,374,374
BEGIN DESCRIPTION:
Catlett Creek 77.9
END DESCRIPTION:
XS GIS Cut Line= 3
      2250481.98      7153914.31      2250139.35      7153516.49
      2249733.01      7152877.35
#Sta/Elev= 30
  4408.2  963.34  4411.2  963.34  4469.8  959.54  4477.5  956.75  4498.4  957.84
  4506.0  955.21  4533.5  952.88  4619.0  949.57  4625.6  952.27  4647.6  953.18
  4676.1  949.52  4696.9  942.36  4717.8  949.84  4759.5  949.71  4803.4  951.95
  4846.2  949.24  4916.0  950.61  4960.3  949.30  4975.5  945.34  4993.4  936.40
  4994.5  935.90  4999.9  936.40  5015.6  945.51  5033.1  947.77  5242.3  945.50
  5357.4  949.62  5466.7  956.67  5509.7  956.95  5560.7  963.60  5690.6  971.54
#Mann=7,-1,0
  4408.2    0.05       0  4411.2    0.12       0  4759.5    0.05       0
  4916.0    0.12       0  4993.4    0.07       0  4999.9    0.12       0
  5015.6    0.05       0
#XS Ineff=2,0
    0.00 4867.60  958.12               0
Permanent Ineff=
       F       F
Bank Sta=4993.4,4999.9
Exp/Cntr=0.3,0.1

Type RM Length L Ch R = 1,67568,119,119,119
BEGIN DESCRIPTION:
Catlett Creek 77.8
END DESCRIPTION:
XS GIS Cut Line= 3
      2250642.24      7153750.83      2250178.79      7153134.92
      2249885.52      7152757.71
#Sta/Elev= 30
  4229.2  956.54  4395.9  948.85  4560.4  946.47  4589.5  940.46  4595.8  944.15
  4604.1  943.69  4610.4  946.24  4624.9  944.56  4631.2  946.49  4674.9  945.52
  4781.1  948.55  4918.5  946.69  4939.4  945.21  4945.6  940.61  4954.0  940.52
  4960.2  937.20  4974.8  935.97  4989.4  937.89  4992.3  935.31  4993.4  934.81
  4998.9  935.31  5039.1  941.57  5045.5  945.83  5060.0  945.64  5068.1  942.66
  5082.2  946.37  5138.7  947.03  5317.0  957.65  5352.3  957.02  5477.8  963.47
#Mann=3,-1,0
  4229.2    0.05       0  4992.3   0.033       0  4998.9    0.05       0
#XS Ineff=2,0
    0.00 4763.90  953.86               0
Permanent Ineff=
       F       F
Bank Sta=4992.3,4998.9
Exp/Cntr=0.3,0.1

Type RM Length L Ch R = 1,67449,358,358,358
BEGIN DESCRIPTION:
Catlett Creek 77.7
END DESCRIPTION:
XS GIS Cut Line= 3
      2250681.97      7153742.96      2250241.30      7153037.24
      2249947.04      7152593.92
#Sta/Elev= 30
  4168.0  956.13  4374.8  947.46  4521.1  946.23  4548.8  941.69  4563.5  945.41
  4630.8  946.99  4636.7  944.46  4919.8  944.02  4971.7  942.39  4994.2  932.27
  4995.2  931.77  5000.8  932.27  5035.0  943.73  5107.2  949.52  5173.3  950.28
  5260.6  956.82  5281.6  954.79  5287.6  957.45  5302.6  957.54  5317.7  955.32
  5323.7  959.41  5332.7  955.99  5338.7  958.74  5353.8  954.33  5359.8  956.06
  5374.8  952.52  5425.9  959.36  5453.0  958.67  5476.8  965.62  5532.1  970.24
#Mann=3,-1,0
  4168.0    0.05       0  4994.2   0.033       0  5000.8    0.05       0
#XS Ineff=2,0
    0.00 4624.50  956.91 5300.00    0.00  960.00
Permanent Ineff=
       F       F
Bank Sta=4994.2,5000.8
Exp/Cntr=0.3,0.1

Type RM Length L Ch R = 1,67091,552,552,552
BEGIN DESCRIPTION:
Catlett Creek 77.6
END DESCRIPTION:
XS GIS Cut Line= 3
      2250983.23      7153564.59      2250528.68      7152932.08
      2250277.52      7152569.83
#Sta/Elev= 30
  4221.1  950.53  4276.7  947.79  4513.6  942.44  4629.0  943.11  4649.9  939.24
  4657.8  939.90  4664.6  942.55  4679.3  943.61  4735.8  942.55  4750.5  939.85
  4771.4  942.70  4865.9  939.77  4953.7  940.12  4972.8  940.45  4978.9  939.03
  4987.5  932.61  4993.6  933.65  5005.1  931.20  5006.2  930.70  5011.7  931.20
  5014.7  937.78  5023.3  942.17  5065.2  940.02  5149.5  941.79  5217.1  945.33
  5345.5  956.60  5390.1  957.20  5396.2  958.90  5417.1  959.45  5440.8  958.60
#Mann=5,-1,0
  4221.1    0.05       0  4953.7    0.12       0  5005.1    0.07       0
  5011.7    0.12       0  5149.5    0.05       0
#XS Ineff=2,0
    0.00 4690.00  950.88               0
Permanent Ineff=
       F       F
Bank Sta=5005.1,5011.7
Exp/Cntr=0.3,0.1

Type RM Length L Ch R = 1,66539,522,522,522
BEGIN DESCRIPTION:
Catlett Creek 77.5
END DESCRIPTION:
XS GIS Cut Line= 3
      2251198.05      7153218.19      2250739.78      7152491.41
      2250547.96      7152153.45
#Sta/Elev= 30
  4140.8  957.93  4356.0  948.59  4465.4  941.28  4538.4  938.78  4617.3  939.34
  4638.5  934.98  4647.0  935.14  4659.7  938.81  4669.0  939.06  4717.9  936.97
  4805.6  938.23  4946.0  937.15  4966.2  937.17  4972.7  935.02  4978.6  929.39
  4994.5  926.18  4995.6  925.68  5001.2  926.18  5009.5  926.74  5015.3  930.71
  5024.6  930.70  5031.2  936.11  5036.9  939.09  5123.0  949.21  5155.2  951.87
  5171.1  955.06  5235.9  958.27  5251.8  960.57  5346.6  962.29  5388.6  965.26
#Mann=5,-1,0
  4140.8    0.05       0  4946.0    0.12       0  4994.5    0.07       0
  5001.2    0.12       0  5123.0    0.05       0
Bank Sta=4994.5,5001.2
Exp/Cntr=0.3,0.1

Type RM Length L Ch R = 1,66017,214,214,214
BEGIN DESCRIPTION:
Catlett Creek 77.0
END DESCRIPTION:
XS GIS Cut Line= 3
      2251379.00      7153010.01      2251162.40      7152276.83
      2251009.53      7151894.25
#Sta/Elev= 30
  4235.5  953.23  4357.2  946.51  4429.0  940.91  4539.3  936.18  4605.9  935.00
  4840.3  934.32  4849.3  934.01  4861.1  927.59  4871.6  931.21  4888.4  933.69
  4934.1  935.07  4959.6  933.84  4975.8  934.47  4986.3  932.66  4992.9  925.37
  4997.2  923.14  5002.6  922.78  5003.9  922.28  5012.2  922.78  5017.7  925.19
  5028.9  935.10  5047.3  936.76  5052.7  936.32  5061.2  937.81  5076.9  937.69
  5110.9  940.08  5262.8  950.52  5292.4  951.54  5316.7  953.69  5412.0  959.09
#Mann=5,-1,0
  4235.5    0.05       0  4888.4    0.12       0  5002.6    0.07       0
  5012.2    0.12       0  5110.9    0.05       0
Bank Sta=5002.6,5012.2
Exp/Cntr=0.3,0.1

Type RM Length L Ch R = 1,65803,185,185,185
BEGIN DESCRIPTION:
Mapping XS 6edc05ca
END DESCRIPTION:
XS GIS Cut Line= 2
      2251554.56      7152663.22      2251169.51      7151797.48
#Sta/Elev= 30
  4523.9  936.79  4615.0  934.52  4658.8  934.38  4735.4  932.87  4772.5  933.56
  4833.9  931.94  4855.8  933.25  4888.6  932.33  4946.2  933.04  4964.0  934.04
  4969.4  933.27  4976.1  925.27  4982.3  921.69  4983.6  921.19  4991.9  921.69
  4992.7  926.55  4998.2  929.80  5015.3  933.81  5039.2  932.93  5091.2  934.25
  5143.4  938.13  5212.9  942.66  5218.3  943.64  5236.1  943.96  5316.8  949.34
  5370.1  950.88  5381.1  950.59  5386.5  951.58  5446.8  953.18  5471.4  955.50
#Mann=5,-1,0
  4523.9    0.05       0  4982.3   0.033       0  4991.9    0.05       0
  5015.3    0.12       0  5143.4    0.05       0
Bank Sta=4982.3,4991.9
Exp/Cntr=0.3,0.1

Type RM Length L Ch R = 1,65618,370,370,370
BEGIN DESCRIPTION:
Mapping XS 7361a016
END DESCRIPTION:
XS GIS Cut Line= 2
      2251715.21      7152581.45      2251341.55      7151764.67
#Sta/Elev= 30
  4541.6  935.85  4638.7  934.79  4675.2  933.26  4774.1  932.03  4833.8  932.30
  4851.1  931.11  4885.3  931.32  4902.8  930.68  4961.1  932.63  4977.4  930.77
  4989.3  919.12  4990.6  918.62  4998.9  919.12  5000.4  923.11  5005.9  927.41
  5016.1  932.32  5023.4  933.66  5038.1  931.87  5046.4  931.67  5092.5  931.32
  5144.0  932.05  5247.0  937.78  5264.6  938.11  5270.1  939.03  5316.1  939.10
  5346.0  941.73  5370.1  942.37  5379.0  942.48  5390.6  944.11  5439.8  946.01
#Mann=4,-1,0
  4541.6    0.05       0  4989.3   0.033       0  4998.9    0.05       0
  5370.1    0.12       0
Bank Sta=4989.3,4998.9
Exp/Cntr=0.3,0.1

Type RM Length L Ch R = 1,65248,626,626,626
BEGIN DESCRIPTION:
Catlett Creek 75.0
END DESCRIPTION:
XS GIS Cut Line= 3
      2252425.88      7152364.78      2251778.86      7151954.94
      2251183.81      7151567.98
#Sta/Elev= 30
  4234.1  961.93  4259.8  960.08  4329.1  955.86  4487.2  943.44  4626.5  932.46
  4668.9  930.52  4867.7  929.52  4929.9  931.32  4966.4  929.98  4975.7  924.74
  4981.6  925.59  4994.6  918.13  4996.1  917.63  5005.2  918.13  5017.1  928.49
  5018.0  929.36  5023.9  926.23  5033.1  931.00  5039.1  929.33  5060.2  930.86
  5151.4  930.08  5214.3  931.22  5226.5  932.83  5386.3  939.53  5546.4  948.64
  5655.1  952.25  5661.1  951.59  5691.3  954.00  5697.3  952.58  5709.8  953.16
#Mann=8,-1,0
  4234.1    0.05       0  4259.8    0.12       0  4487.2    0.05       0
  4867.7    0.12       0  4994.6    0.07       0  5005.2    0.12       0
  5017.1    0.05       0  5151.4    0.12       0
Bank Sta=4994.6,5005.2
Exp/Cntr=0.3,0.1

Type RM Length L Ch R = 1,64622,558,558,558
BEGIN DESCRIPTION:
Catlett Creek 74.0
END DESCRIPTION:
XS GIS Cut Line= 3
      2252571.65      7152187.65      2252179.00      7151760.00
      2251975.77      7151487.01
#Sta/Elev= 30
  4419.7  956.56  4441.3  955.09  4448.1  955.71  4469.7  953.56  4490.7  953.46
  4498.0  951.93  4575.8  946.17  4639.3  943.65  4697.7  939.61  4731.1  938.22
  4823.6  928.10  4844.6  926.95  4901.3  926.23  4964.8  927.92  4979.0  926.10
  4986.4  921.60  4993.2  921.52  4996.9  917.31  5002.1  916.14  5003.6  915.64
  5013.0  916.14  5028.4  928.04  5036.8  928.53  5199.7  928.47  5249.6  926.96
  5293.2  928.17  5314.1  928.79  5322.5  934.52  5328.7  935.75  5340.6  935.75
#Mann=5,-1,0
  4419.7    0.05       0  4697.7    0.12       0  5002.1    0.07       0
  5013.0    0.12       0  5293.2    0.05       0
Bank Sta=5002.1,5013
Exp/Cntr=0.3,0.1

Type RM Length L Ch R = 1,64064,647,647,647
BEGIN DESCRIPTION:
Mapping XS 93f405ac
END DESCRIPTION:
XS GIS Cut Line= 2
      2252857.27      7151549.24      2251899.82      7151084.91
#Sta/Elev= 30
  4388.0  944.75  4513.1  938.73  4530.1  935.70  4558.2  934.87  4580.8  931.66
  4658.9  926.49  4699.2  923.99  4789.5  922.86  4857.2  924.93  4896.8  923.54
  4925.0  925.04  4970.1  925.14  4975.7  923.53  4986.2  918.09  4987.2  914.90
  4988.7  914.40  4998.2  914.90  5009.1  919.39  5015.2  924.08  5020.8  925.74
  5052.9  924.67  5065.9  923.04  5088.5  923.04  5141.8  925.04  5186.3  924.96
  5230.7  927.13  5269.1  925.93  5336.1  927.57  5342.4  929.17  5452.1  939.79
#Mann=6,-1,0
  4388.0    0.05       0  4658.9    0.12       0  4987.2    0.07       0
  4998.2    0.12       0  5009.1    0.05       0  5336.1    0.12       0
Bank Sta=4987.2,4998.2
Exp/Cntr=0.3,0.1

Type RM Length L Ch R = 1,63417,602,602,602
BEGIN DESCRIPTION:
Mapping XS 2efc0744
END DESCRIPTION:
XS GIS Cut Line= 3
      2252879.55      7150995.07      2252643.28      7150897.14
      2251738.77      7150829.57
#Sta/Elev= 30
  4837.5  939.90  4859.1  940.04  4928.2  936.03  4935.5  934.73  4941.5  932.35
  4947.0  932.00  4957.2  924.81  4965.4  914.50  4973.3  911.50  4974.8  911.00
  4984.3  911.50  4989.3  914.78  4994.7  915.73  5000.5  919.47  5018.6  921.84
  5177.8  920.10  5249.2  920.43  5308.1  919.54  5378.3  921.10  5448.5  919.53
  5512.5  920.84  5548.8  921.09  5558.8  920.36  5568.9  922.07  5609.0  922.84
  5639.1  926.11  5669.1  926.79  5699.2  928.72  5926.1  946.80  6000.3  951.92
#Mann=6,-1,0
  4837.5    0.05       0  4928.2    0.12       0  4973.3    0.07       0
  4984.3    0.12       0  5249.2    0.05       0  5512.5    0.12       0
Bank Sta=4973.3,4984.3
Exp/Cntr=0.3,0.1

Type RM Length L Ch R = 1,62815,361,361,361
BEGIN DESCRIPTION:
Catlett Creek 71.0
END DESCRIPTION:
XS GIS Cut Line= 3
      2252879.02      7150810.01      2252579.00      7150560.00
      2252179.03      7150210.03
#Sta/Elev= 30
  4608.9  932.14  4636.9  930.82  4687.0  924.59  4715.0  922.52  4811.0  917.98
  4864.7  916.82  4907.7  918.21  4957.1  918.22  4985.8  916.25  4992.3  914.85
  4996.2  911.54  5002.8  911.54  5007.7  908.73  5009.2  908.23  5018.7  908.73
  5019.4  911.27  5020.8  916.36  5027.4  917.93  5098.6  917.79  5148.0  915.73
  5162.2  916.00  5176.4  914.21  5290.3  916.92  5297.0  916.09  5325.5  918.60
  5346.3  918.61  5417.5  922.85  5446.0  927.40  5509.6  930.63  5530.9  933.16
#Mann=5,-1,0
  4608.9    0.05       0  4811.0    0.12       0  5007.7    0.07       0
  5018.7    0.12       0  5019.4    0.05       0
Bank Sta=5007.7,5018.7
Exp/Cntr=0.3,0.1

Type RM Length L Ch R = 1,62454,580,580,580
BEGIN DESCRIPTION:
Catlett Creek 70.0
END DESCRIPTION:
XS GIS Cut Line= 3
      2253279.02      7150660.02      2252768.90      7150270.39
      2252116.06      7150028.24
#Sta/Elev= 30
  4358.1  929.37  4465.1  921.54  4600.1  915.88  4650.1  914.08  4679.2  914.28
  4693.7  915.75  4729.1  914.86  4814.3  915.57  4828.8  914.30  4843.4  914.41
  4848.1  915.45  4914.1  914.91  4942.5  915.85  4960.7  915.83  4986.7  914.01
  4996.8  910.11  5002.6  910.11  5004.9  907.14  5006.4  906.64  5015.9  907.14
  5021.2  914.21  5031.9  915.05  5351.9  914.84  5383.9  916.77  5450.0  917.58
  5535.8  922.71  5560.8  925.80  5566.2  924.82  5646.6  929.62  5696.3  930.65
#Mann=7,-1,0
  4358.1    0.05       0  4600.1    0.12       0  4848.1    0.05       0
  4942.5    0.12       0  4960.7    0.05       0  5004.9   0.033       0
  5015.9    0.05       0
Bank Sta=5004.9,5015.9
Exp/Cntr=0.3,0.1

Type RM Length L Ch R = 1,61874,929,929,929
BEGIN DESCRIPTION:
Catlett Creek 69.0
END DESCRIPTION:
XS GIS Cut Line= 3
      2253524.39      7150590.29      2253227.03      7150104.35
      2252703.38      7149530.86
#Sta/Elev= 30
  4430.3  936.32  4559.5  930.31  4617.5  925.06  4660.1  918.88  4761.6  913.64
  4944.5  913.17  4950.3  908.46  4965.8  909.69  4971.6  905.06  4987.1  906.59
  5008.6  906.31  5010.4  904.92  5012.0  904.42  5021.5  904.92  5022.8  911.18
  5030.2  910.22  5037.0  912.89  5114.9  914.38  5249.6  912.92  5256.5  911.26
  5263.3  913.18  5270.7  910.75  5277.5  912.14  5284.9  909.86  5291.7  910.98
  5334.2  905.19  5348.4  906.24  5370.0  912.41  5419.3  916.29  5776.6  925.46
#Mann=5,-1,0
  4430.3    0.05       0  4761.6    0.12       0  5010.4    0.07       0
  5021.5    0.12       0  5114.9    0.05       0
Bank Sta=5010.4,5021.5
Exp/Cntr=0.3,0.1
