HEC-RAS study Catlett Creek.prj: Catlett Creek Base Level Engineering

--- Catlett Creek.g01 (geometry) --- (continued)

Type RM Length L Ch R = 1,60945,511,511,511
BEGIN DESCRIPTION:
Catlett Creek 68.0
END DESCRIPTION:
XS GIS Cut Line= 3
      2253684.97      7150542.50      2253384.92      7149668.47
      2253372.46      7149379.84
#Sta/Elev= 30
  4075.9  936.02  4099.7  933.77  4120.8  929.79  4194.8  927.39  4263.6  921.70
  4357.4  917.54  4364.0  916.19  4414.6  914.72  4459.2  911.92  4560.5  910.38
  4586.0  912.00  4628.1  912.16  4670.6  910.43  4681.2  911.70  4784.4  910.89
  4860.9  910.99  4871.5  911.93  4883.5  910.57  4934.9  909.66  4946.0  910.94
  4966.7  904.67  4972.0  905.67  4977.3  904.33  5000.0  904.30  5011.8  901.81
  5013.3  901.31  5023.1  901.81  5048.5  918.64  5078.5  922.59  5288.9  925.19
#Mann=4,-1,0
  4075.9    0.05       0  4560.5    0.12       0  5011.8    0.07       0
  5023.1    0.12       0
Bank Sta=5011.8,5023.1
Exp/Cntr=0.3,0.1

Type RM Length L Ch R = 1,60434,357,357,357
BEGIN DESCRIPTION:
Catlett Creek 67.0
END DESCRIPTION:
XS GIS Cut Line= 3
      2254060.10      7150144.29      2253828.36      7149659.65
      2253578.98      7149259.97
#Sta/Elev= 30
  4462.8  931.35  4475.0  931.12  4511.9  926.43  4543.0  925.83  4653.6  917.34
  4744.7  909.91  4826.2  908.64  4843.4  905.34  4848.9  906.69  4855.5  905.03
  4866.0  905.64  4871.6  907.44  4910.9  908.93  4939.6  906.96  4945.1  908.24
  4977.4  903.14  4984.8  900.71  4986.4  900.21  4996.2  900.71  5002.7  900.88
  5006.9  903.67  5022.2  908.16  5028.1  907.45  5049.3  909.53  5122.5  908.13
  5232.2  908.95  5305.3  914.67  5363.1  920.50  5369.0  922.21  5471.1  929.90
#Mann=4,-1,0
  4462.8    0.05       0  4653.6    0.12       0  4984.8    0.07       0
  4996.2    0.12       0
Bank Sta=4984.8,4996.2
Exp/Cntr=0.3,0.1

Type RM Length L Ch R = 1,60077,965,965,965
BEGIN DESCRIPTION:
Catlett Creek 66.0
END DESCRIPTION:
XS GIS Cut Line= 3
      2254236.20      7150071.62      2254115.05      7149523.14
      2253690.74      7149076.16
#Sta/Elev= 30
  4438.3  933.30  4495.6  930.59  4675.9  918.40  4757.4  913.67  4767.7  912.02
  4772.9  909.75  4849.6  904.45  4957.8  908.32  4972.5  903.93  4993.0  901.93
  4993.3  900.27  4994.9  899.77  5004.7  900.27  5006.4  902.47  5013.6  904.07
  5041.9  907.65  5155.2  905.63  5247.0  907.24  5268.1  909.88  5317.8  910.30
  5324.7  909.02  5367.2  909.85  5543.9  925.72  5551.2  924.54  5558.1  926.16
  5565.4  925.13  5572.3  927.71  5593.7  930.11  5607.8  929.71  5616.3  932.36
#Mann=4,-1,0
  4438.3    0.05       0  4675.9    0.12       0  4993.3    0.07       0
  5004.7    0.12       0
Bank Sta=4993.3,5004.7
Exp/Cntr=0.3,0.1

Type RM Length L Ch R = 1,59112,454,454,454
BEGIN DESCRIPTION:
Catlett Creek 65.0
END DESCRIPTION:
XS GIS Cut Line= 3
      2254288.28      7149995.67      2254729.00      7148860.00
      2254739.58      7148604.61
#Sta/Elev= 30
  3781.7  932.46  3795.3  930.03  3948.7  924.55  4013.0  919.60  4127.4  906.60
  4211.8  903.78  4549.4  902.28  4667.4  905.38  4677.4  902.92  4682.7  905.08
  4688.8  902.76  4721.0  902.41  4731.7  902.58  4737.2  905.94  4742.6  902.50
  4785.4  903.08  4791.7  905.71  4797.0  902.43  4806.8  905.46  4885.8  902.58
  4967.7  903.73  4984.9  901.63  4990.3  903.36  4997.2  898.84  5004.1  897.99
  5005.7  897.49  5015.6  897.99  5029.9  918.25  5150.0  925.57  5255.5  926.73
#Mann=4,-1,0
  3781.7    0.05       0  4885.8    0.12       0  5004.1    0.07       0
  5015.6    0.12       0
Bank Sta=5004.1,5015.6
Exp/Cntr=0.3,0.1

Type RM Length L Ch R = 1,58658,494,494,494
BEGIN DESCRIPTION:
Catlett Creek 64.0
END DESCRIPTION:
XS GIS Cut Line= 5
      2254299.15      7149999.98      2254483.59      7149689.68
      2254916.17      7149127.11      2254973.97      7148796.27
      2254877.38      7148626.97
#Sta/Elev= 30
  3927.9  931.86  4160.5  917.54  4206.3  913.92  4255.0  908.39  4350.2  904.08
  4805.7  901.24  4834.1  901.33  4842.3  903.39  4856.1  903.82  4863.1  903.68
  4869.4  901.99  4877.6  904.04  4883.9  901.12  4956.4  903.19  4983.6  901.47
  4986.0  898.43  4987.6  897.93  4997.5  898.43  5005.7  898.63  5015.9  901.11
  5042.7  901.96  5056.4  901.19  5087.0  902.97  5107.3  902.22  5137.7  904.55
  5156.6  907.42  5161.7  906.90  5216.1  910.78  5341.6  917.07  5529.3  931.84
#Mann=4,-1,0
  3927.9    0.05       0  4986.0   0.033       0  4997.5    0.05       0
  5056.4    0.12       0
Bank Sta=4986,4997.5
Exp/Cntr=0.3,0.1

Type RM Length L Ch R = 1,58164,459,459,459
BEGIN DESCRIPTION:
Catlett Creek 63.0
END DESCRIPTION:
XS GIS Cut Line= 3
      2256308.68      7149572.49      2255229.00      7148810.00
      2254904.01      7148535.01
#Sta/Elev= 30
  3682.3  938.67  3755.4  937.14  3864.0  932.50  3905.8  929.71  3971.1  921.99
  4063.4  916.77  4107.8  915.79  4214.9  909.42  4488.2  901.73  4583.0  901.87
  4610.1  902.30  4642.1  898.81  4654.7  898.42  4656.4  897.92  4666.5  898.42
  4732.0  901.14  4860.0  902.18  4868.7  900.66  4881.7  901.46  4918.4  900.33
  4967.3  900.65  4975.8  901.93  4990.6  899.24  5011.2  898.56  5054.1  901.11
  5210.1  915.09  5328.9  924.19  5401.2  928.67  5409.0  930.22  5429.8  929.98
#Mann=6,-1,0
  3682.3    0.05       0  4583.0    0.12       0  4642.1    0.05       0
  4654.7   0.033       0  4666.5    0.05       0  5328.9    0.12       0
Bank Sta=4654.7,4666.5
Exp/Cntr=0.3,0.1

Type RM Length L Ch R = 1,57705,455,455,455
BEGIN DESCRIPTION:
Catlett Creek 62.0
END DESCRIPTION:
XS GIS Cut Line= 3
      2256397.63      7149051.64      2255520.90      7148466.07
      2254953.96      7148184.98
#Sta/Elev= 30
  3945.7  931.22  4148.5  925.21  4206.2  924.99  4220.6  926.35  4248.2  925.37
  4284.3  926.79  4314.3  925.17  4328.9  926.13  4335.3  924.69  4356.3  925.87
  4413.4  924.42  4443.4  922.94  4494.5  916.50  4551.6  915.77  4581.4  912.04
  4602.6  910.75  4608.6  911.35  4623.7  907.83  4629.7  908.89  4659.7  904.57
  4731.8  898.81  5262.5  897.97  5264.2  897.47  5274.4  897.97  5358.2  905.92
  5453.4  912.70  5544.2  921.14  5587.9  924.49  5616.0  927.97  5632.8  928.29
#Mann=4,-1,0
  3945.7    0.05       0  5262.5   0.033       0  5274.4    0.05       0
  5544.2    0.12       0
Bank Sta=5262.5,5274.4
Exp/Cntr=0.3,0.1

Type RM Length L Ch R = 1,57250,444,444,444
BEGIN DESCRIPTION:
Catlett Creek 61.0
END DESCRIPTION:
XS GIS Cut Line= 3
      2256623.36      7149051.67      2255628.46      7148044.78
      2255129.04      7147760.02
#Sta/Elev= 30
  3584.5  933.89  3624.1  931.96  3857.4  928.02  4027.2  927.51  4161.6  925.83
  4253.4  921.48  4267.6  921.53  4324.2  917.94  4437.3  912.69  4465.6  912.36
  4508.0  908.93  4515.0  907.60  4635.3  899.45  4643.5  898.06  4645.1  897.56
  4655.4  898.06  4833.3  898.82  5229.6  898.53  5244.3  899.26  5252.6  901.09
  5303.4  906.34  5319.3  908.98  5325.0  908.66  5362.5  913.03  5384.1  913.88
  5399.9  916.20  5421.5  917.87  5494.4  927.51  5508.0  930.35  5574.9  935.56
#Mann=3,-1,0
  3584.5    0.05       0  4643.5   0.033       0  4655.4    0.05       0
Bank Sta=4643.5,4655.4
Exp/Cntr=0.3,0.1

Type RM Length L Ch R = 1,56806,488,488,488
BEGIN DESCRIPTION:
Catlett Creek 60.0
END DESCRIPTION:
XS GIS Cut Line= 3
      2256794.81      7149027.81      2255776.49      7147653.96
      2255179.03      7147160.02
#Sta/Elev= 30
  3289.9  930.56  3307.0  929.33  3442.6  929.35  3793.2  925.73  4035.2  925.55
  4099.9  924.55  4164.6  922.55  4264.8  917.68  4285.6  915.75  4400.4  914.52
  4465.1  904.30  4536.1  900.57  4550.7  898.19  4571.5  899.02  4600.8  898.20
  4621.6  898.96  5222.8  898.14  5224.5  897.64  5234.7  898.14  5292.6  899.39
  5356.4  905.21  5441.1  915.03  5469.8  918.98  5484.1  922.30  5554.7  930.75
  5562.3  932.58  5597.4  934.84  5640.4  939.57  5661.2  940.26  5775.2  952.30
#Mann=3,-1,0
  3289.9    0.05       0  5222.8   0.033       0  5234.7    0.05       0
Bank Sta=5222.8,5234.7
Exp/Cntr=0.3,0.1

Type RM Length L Ch R = 1,56318,149,149,149
BEGIN DESCRIPTION:
Catlett Creek 59.0
END DESCRIPTION:
XS GIS Cut Line= 3
      2256967.38      7148457.62      2256085.12      7147312.72
      2255377.81      7146709.66
#Sta/Elev= 30
  3554.6  922.98  3708.5  921.86  3872.5  917.09  3951.3  912.80  4021.9  910.67
  4100.8  904.66  4258.4  898.22  4636.6  897.91  4638.2  897.41  4648.5  897.91
  5027.5  898.93  5084.6  897.98  5098.9  899.42  5105.5  901.53  5148.3  904.58
  5169.2  909.13  5197.7  911.59  5212.0  911.02  5232.8  913.85  5290.0  916.13
  5453.6  915.87  5474.4  916.96  5488.7  922.98  5503.0  927.26  5560.0  925.48
  5644.6  928.67  5658.9  927.62  5722.6  928.17  5857.6  932.29  5929.5  932.96
#Mann=3,-1,0
  3554.6    0.05       0  4636.6   0.033       0  4648.5    0.05       0
Bank Sta=4636.6,4648.5
Exp/Cntr=0.3,0.1

Type RM Length L Ch R = 1,56169,191,191,191
BEGIN DESCRIPTION:
Catlett Creek 58.5
END DESCRIPTION:
XS GIS Cut Line= 5
      2257188.63      7148443.77      2256201.85      7147231.42
      2256037.49      7147031.48      2255961.19      7146785.81
      2255669.23      7146439.26
#Sta/Elev= 30
  3440.9  919.07  3563.7  922.21  3699.4  920.59  3705.9  922.53  3792.1  922.38
  3812.9  920.15  3827.3  922.58  3862.5  920.96  3934.3  922.77  3940.7  920.06
  3955.1  922.84  4004.7  921.21  4012.6  922.87  4019.0  920.95  4033.4  922.95
  4082.9  921.29  4097.3  923.12  4360.9  923.61  4367.3  921.91  4374.1  923.77
  4594.3  924.06  5266.3  921.92  5298.8  916.17  5300.4  915.67  5310.7  916.17
  5472.8  917.61  5505.3  921.84  5561.4  919.68  5788.9  925.01  5973.3  926.26
#Mann=3,-1,0
  3440.9    0.05       0  5298.8   0.033       0  5310.7    0.05       0
Bank Sta=5298.8,5310.7
Exp/Cntr=0.3,0.1

Type RM Length L Ch R = 1,55978,533,533,533
BEGIN DESCRIPTION:
Catlett Creek 58.0
END DESCRIPTION:
XS GIS Cut Line= 4
      2257039.70      7147793.63      2256275.50      7147061.15
      2256178.49      7146730.12      2255756.76      7146446.38
#Sta/Elev= 30
  4016.4  906.50  4090.1  904.14  4139.8  898.06  4189.2  895.00  4394.2  887.26
  4896.5  887.35  4924.8  882.95  4954.0  871.78  4955.7  871.28  4965.9  871.78
  5002.4  872.19  5009.7  877.90  5077.6  886.90  5080.8  892.46  5159.5  893.91
  5186.3  885.35  5191.5  887.23  5363.7  887.08  5388.8  890.13  5409.6  897.12
  5448.2  896.19  5499.2  900.29  5520.2  899.94  5535.2  903.00  5571.2  905.88
  5592.2  905.33  5643.2  912.18  5700.2  914.35  5715.1  917.08  5928.2  921.77
#Mann=3,-1,0
  4016.4    0.05       0  4954.0   0.033       0  4965.9    0.05       0
Bank Sta=4954,4965.9
Exp/Cntr=0.3,0.1

Type RM Length L Ch R = 1,55445,218,218,218
BEGIN DESCRIPTION:
Catlett Creek 57.0
END DESCRIPTION:
XS GIS Cut Line= 3
      2257148.37      7147284.12      2256379.00      7146610.00
      2255804.69      7146304.99
#Sta/Elev= 30
  3981.6  885.06  4445.1  883.42  4635.8  885.04  4898.2  884.02  4926.2  882.74
  4933.8  878.47  4940.5  877.37  4948.1  872.57  4970.6  870.90  4972.2  870.40
  4982.5  870.90  4990.8  873.66  5007.4  874.73  5034.7  880.71  5049.8  881.49
  5062.3  884.00  5100.6  882.75  5197.0  886.12  5242.3  888.95  5270.8  892.52
  5353.1  897.88  5358.7  897.15  5375.1  900.47  5424.7  903.40  5441.0  905.92
  5567.3  911.93  5572.9  909.25  5582.0  909.08  5604.6  913.24  5654.8  915.77
#Mann=3,-1,0
  3981.6    0.05       0  4970.6   0.033       0  4982.5    0.05       0
Bank Sta=4970.6,4982.5
Exp/Cntr=0.3,0.1

Type RM Length L Ch R = 1,55227,110,110,110
BEGIN DESCRIPTION:
Catlett Creek 56.5
END DESCRIPTION:
XS GIS Cut Line= 3
      2257205.50      7146923.61      2256458.74      7146414.31
      2255957.94      7146124.71
#Sta/Elev= 30
  4096.1  891.12  4110.7  889.89  4182.5  890.74  4326.1  888.63  4427.8  885.72
  4448.8  886.05  4463.7  884.61  4484.7  885.03  4535.5  882.79  4664.2  881.69
  4694.0  880.93  4744.9  877.52  4924.4  875.85  4939.2  877.58  4960.3  876.73
  4966.3  877.73  4981.3  874.25  4987.6  870.98  4993.4  869.45  4995.0  868.95
  5005.4  869.45  5017.8  874.25  5045.9  878.20  5082.4  879.74  5104.0  882.23
  5184.5  884.22  5230.7  886.73  5333.6  895.75  5398.2  898.14  5578.5  911.10
#Mann=3,-1,0
  4096.1    0.05       0  4993.4   0.033       0  5005.4    0.05       0
Bank Sta=4993.4,5005.4
Exp/Cntr=0.3,0.1

Type RM Length L Ch R = 1,55117,416,416,416
BEGIN DESCRIPTION:
Catlett Creek 56.0
END DESCRIPTION:
XS GIS Cut Line= 3
      2257188.27      7146744.61      2256509.47      7146317.10
      2256044.25      7146014.83
#Sta/Elev= 30
  4197.8  897.95  4215.2  895.68  4221.2  896.99  4251.7  895.82  4272.9  897.17
  4288.2  895.42  4294.1  896.78  4309.4  894.69  4315.3  896.03  4324.7  894.62
  4330.6  895.74  4613.2  880.32  4838.0  880.62  4947.5  879.06  4984.0  872.61
  4989.9  867.03  4991.3  866.87  4993.0  866.37  5003.3  866.87  5048.3  874.17
  5056.6  877.57  5062.5  874.34  5071.7  880.58  5280.0  888.86  5295.1  894.06
  5352.5  898.69  5373.6  901.58  5388.7  901.12  5467.2  908.56  5554.8  914.38
#Mann=3,-1,0
  4197.8    0.05       0  4991.3   0.033       0  5003.3    0.05       0
Bank Sta=4991.3,5003.3
Exp/Cntr=0.3,0.1

Type RM Length L Ch R = 1,54701,875,875,875
BEGIN DESCRIPTION:
Catlett Creek 55.0
END DESCRIPTION:
XS GIS Cut Line= 3
      2257068.92      7146200.99      2256612.11      7145926.57
      2256305.07      7145836.43
#Sta/Elev= 30
  4467.1  889.49  4534.1  885.38  4561.3  882.10  4576.8  881.13  4592.4  878.41
  4656.5  877.65  4677.9  879.95  4693.4  878.22  4723.6  878.65  4730.3  879.86
  4736.2  878.84  4745.9  879.83  4794.5  878.32  4852.8  879.17  4926.6  878.28
  4948.0  879.13  4969.3  874.56  4979.0  869.99  4992.9  865.56  4994.5  865.06
  5004.9  865.56  5013.7  873.30  5026.4  877.35  5086.6  880.24  5126.9  883.71
  5145.8  886.27  5184.4  888.73  5251.1  894.76  5289.7  896.03  5320.0  898.28
#Mann=5,-1,0
  4467.1    0.05       0  4992.9   0.033       0  5004.9    0.05       0
  5026.4    0.12       0  5126.9    0.05       0
Bank Sta=4992.9,5004.9
Exp/Cntr=0.3,0.1

Type RM Length L Ch R = 1,53826,307,307,307
BEGIN DESCRIPTION:
Catlett Creek 54.5
END DESCRIPTION:
XS GIS Cut Line= 3
      2257145.41      7145689.03      2256907.30      7145297.00
      2256644.90      7144350.26
#Sta/Elev= 30
  4529.0  889.64  4590.9  887.08  4622.5  888.12  4643.2  888.55  4649.0  886.78
  4664.5  888.27  4670.3  886.04  4701.3  887.05  4707.1  883.87  4722.6  885.58
  4728.5  882.88  4738.1  884.05  4744.0  881.24  4759.4  882.04  4802.1  876.10
  4881.6  877.34  4955.2  875.56  4976.5  865.60  4985.9  865.10  4987.9  864.60
  5003.9  865.10  5005.3  868.77  5034.4  870.31  5057.2  877.01  5129.5  875.19
  5254.4  875.86  5379.3  879.42  5540.8  878.39  5686.0  880.27  5970.1  883.47
#Mann=7,-1,0
  4529.0    0.05       0  4622.5    0.12       0  4985.9    0.07       0
  5003.9    0.12       0  5129.5    0.05       0  5540.8    0.12       0
  5686.0    0.05       0
Bank Sta=4985.9,5003.9
Exp/Cntr=0.3,0.1

Type RM Length L Ch R = 1,53519,560,560,560
BEGIN DESCRIPTION:
Catlett Creek 54.0
END DESCRIPTION:
XS GIS Cut Line= 3
      2257171.44      7145662.97      2257144.47      7145103.33
      2257187.07      7144467.65
#Sta/Elev= 30
  4462.1  890.25  4545.2  891.99  4595.2  895.63  4685.3  886.69  4835.3  873.96
  4855.5  872.34  4885.6  874.73  4935.6  875.09  4965.7  868.94  5005.7  866.25
  5006.7  863.09  5008.7  862.59  5024.8  863.09  5026.6  866.67  5035.8  874.16
  5045.8  876.90  5065.8  877.74  5095.5  876.38  5256.2  875.69  5356.5  877.47
  5416.6  880.72  5446.7  885.19  5467.9  884.53  5486.8  886.76  5498.2  886.95
  5556.9  893.17  5597.0  892.93  5612.8  894.73  5620.3  894.25  5659.5  896.24
#Mann=7,-1,0
  4462.1    0.05       0  4835.3    0.12       0  5006.7    0.07       0
  5024.8    0.12       0  5095.5    0.05       0  5498.2    0.12       0
  5620.3    0.05       0
Bank Sta=5006.7,5024.8
Exp/Cntr=0.3,0.1

Type RM Length L Ch R = 1,52959,606,606,606
BEGIN DESCRIPTION:
Catlett Creek 53.0
END DESCRIPTION:
XS GIS Cut Line= 3
      2257739.38      7145854.18      2257540.41      7145154.31
      2257166.23      7144287.97
#Sta/Elev= 30
  4272.4  890.96  4365.2  882.86  4584.0  874.50  4775.8  871.81  4939.8  873.60
  4948.8  874.25  4987.9  864.08  4990.6  861.91  4992.6  861.41  5008.7  861.91
  5013.2  861.92  5018.6  865.78  5036.7  871.84  5048.3  873.91  5067.9  873.35
  5135.4  872.72  5157.2  874.19  5241.0  870.97  5322.4  873.96  5468.9  874.94
  5597.3  882.20  5690.9  892.71  5702.2  895.56  5749.2  895.85  5772.7  898.61
  5801.7  898.52  5832.6  901.00  5865.2  900.73  5897.8  896.79  5943.7  894.75
#Mann=6,-1,0
  4272.4    0.05       0  4939.8    0.12       0  4990.6    0.07       0
  5008.7    0.12       0  5067.9    0.05       0  5897.8    0.12       0
Bank Sta=4990.6,5008.7
Exp/Cntr=0.3,0.1

Type RM Length L Ch R = 1,52353,596,596,596
BEGIN DESCRIPTION:
Mapping XS 375727cf
END DESCRIPTION:
XS GIS Cut Line= 3
      2258268.29      7146011.85      2258217.69      7145542.98
      2257396.15      7144054.32
#Sta/Elev= 30
  3555.3  882.65  3577.3  881.57  3607.5  878.04  3647.7  875.75  3708.0  874.63
  3738.2  872.50  3858.9  870.00  4116.6  868.10  4144.5  869.02  4588.8  871.93
  4852.7  871.43  4898.2  873.48  4918.2  871.36  4941.8  863.86  4947.5  865.96
  4963.5  861.29  4978.3  860.40  4991.0  861.06  4998.0  857.43  5000.0  856.93
  5016.1  857.43  5028.8  872.21  5219.1  871.30  5286.7  872.51  5435.2  877.32
  5560.6  883.47  5604.1  884.54  5653.4  887.71  5685.5  887.49  5727.2  889.65
#Mann=4,-1,0
  3555.3    0.05       0  4918.2    0.12       0  4998.0    0.07       0
  5016.1    0.05       0
Bank Sta=4998,5016.1
Exp/Cntr=0.3,0.1

Type RM Length L Ch R = 1,51757,302,302,302
BEGIN DESCRIPTION:
Mapping XS 12f821e5
END DESCRIPTION:
XS GIS Cut Line= 2
      2259338.57      7145698.97      2257553.59      7143767.60
#Sta/Elev= 30
  3449.1  879.81  3568.6  870.28  3788.0  869.85  3886.7  866.39  3964.9  868.04
  3985.9  865.98  4000.1  861.28  4004.7  863.05  4033.3  866.26  4113.5  866.09
  4198.0  869.58  4219.5  866.63  4866.1  869.58  4905.6  871.50  4934.0  869.68
  4962.3  863.21  4967.4  855.12  4969.4  854.62  4985.5  855.12  5019.0  862.04
  5026.4  865.86  5068.3  870.64  5104.1  870.03  5125.0  864.36  5139.2  863.96
  5189.1  864.06  5203.3  869.77  5252.2  869.89  5804.3  881.48  6079.0  898.65
#Mann=7,-1,0
  3449.1    0.05       0  4004.7    0.12       0  4033.3    0.05       0
  4866.1    0.12       0  4967.4    0.07       0  4985.5    0.12       0
  5252.2    0.05       0
Bank Sta=4967.4,4985.5
Exp/Cntr=0.3,0.1

Type RM Length L Ch R = 1,51455,1183,1183,1183
BEGIN DESCRIPTION:
Mapping XS 3c7fdfff
END DESCRIPTION:
XS GIS Cut Line= 2
      2259597.31      7145616.85      2257780.42      7143654.51
#Sta/Elev= 30
  3490.5  874.74  3543.5  877.88  3656.9  868.27  3756.1  866.15  4124.1  866.37
  4138.3  863.64  4152.5  856.01  4173.4  854.44  4187.6  862.46  4201.8  865.02
  4768.9  869.04  4830.1  869.65  4866.9  869.76  4963.8  852.71  4965.8  852.21
  4982.0  852.71  5029.6  854.57  5051.1  866.56  5121.6  864.97  5185.5  880.84
  5228.0  874.24  5397.5  874.02  5447.4  881.49  5510.9  883.45  5864.7  887.37
  5978.1  884.46  5999.1  891.02  6020.6  892.86  6077.6  892.58  6164.8  898.38
#Mann=6,-1,0
  3490.5    0.05       0  4768.9    0.12       0  4830.1    0.05       0
  4963.8   0.033       0  4982.0    0.05       0  6077.6    0.12       0
Bank Sta=4963.8,4982
Exp/Cntr=0.3,0.1

Type RM Length L Ch R = 1,50272,592,592,592
BEGIN DESCRIPTION:
Catlett Creek 49.0
END DESCRIPTION:
XS GIS Cut Line= 3
      2259693.26      7145600.04      2259491.47      7144960.00
      2259330.14      7143876.64
#Sta/Elev= 30
  4328.9  875.17  4444.3  868.71  4524.4  868.53  4621.5  865.46  4874.2  862.76
  4916.1  862.79  4960.8  864.73  4979.1  859.39  4987.9  855.22  4993.2  854.00
  4997.4  850.63  5000.8  850.15  5002.8  849.65  5019.5  850.15  5020.2  853.46
  5024.9  855.91  5040.4  862.37  5060.7  864.62  5141.5  863.86  5320.4  865.71
  5374.1  865.00  5586.4  865.62  5606.6  866.42  5788.6  867.73  5839.1  869.08
  5929.2  873.36  6003.6  879.56  6051.5  881.23  6071.6  884.16  6095.3  885.99
#Mann=6,-1,0
  4328.9    0.05       0  4979.1    0.12       0  5000.8    0.07       0
  5019.5    0.12       0  5024.9    0.05       0  6071.6    0.12       0
Bank Sta=5000.8,5019.5
Exp/Cntr=0.3,0.1

Type RM Length L Ch R = 1,49680,669,669,669
BEGIN DESCRIPTION:
Catlett Creek 48.0
END DESCRIPTION:
XS GIS Cut Line= 3
      2260005.88      7145563.01      2260069.78      7144998.72
      2260263.69      7143755.75
#Sta/Elev= 30
  4432.1  876.96  4485.4  874.35  4502.4  872.20  4592.1  867.15  4797.4  860.92
  4861.3  861.03  4946.0  858.65  4968.5  853.88  4978.6  849.62  4979.2  846.83
  4981.2  846.33  4998.0  846.83  5025.7  850.85  5030.7  856.72  5039.2  860.24
  5049.3  862.05  5085.3  861.60  5170.8  860.58  5191.0  861.79  5219.1  860.84
  5287.0  862.01  5322.6  860.83  5464.3  860.16  6003.1  861.28  6133.8  864.49
  6172.7  868.00  6196.6  868.02  6213.2  870.11  6223.3  869.79  6258.0  872.96
#Mann=5,-1,0
  4432.1    0.05       0  4861.3    0.12       0  4979.2    0.07       0
  4998.0    0.12       0  5085.3    0.05       0
Bank Sta=4979.2,4998
Exp/Cntr=0.3,0.1

Type RM Length L Ch R = 1,49011,280,280,280
BEGIN DESCRIPTION:
Catlett Creek 47.0
END DESCRIPTION:
XS GIS Cut Line= 3
      2260570.98      7145622.97      2260529.00      7145160.00
      2260383.65      7143783.42
#Sta/Elev= 30
  4535.2  877.75  4578.3  874.55  4613.0  873.52  4658.7  870.05  4678.8  870.19
  4749.0  865.44  4842.8  862.41  4889.6  861.03  4949.9  861.41  4980.0  851.22
  4988.2  846.97  4990.2  846.47  5007.0  846.97  5020.2  848.63  5040.3  856.41
  5046.5  860.90  5085.8  860.31  5130.8  859.44  5242.3  859.53  5330.1  860.77
  5362.1  859.70  5442.5  860.15  5633.6  859.05  5902.4  859.43  6025.7  860.74
  6066.0  859.87  6136.4  860.30  6196.7  863.25  6247.0  864.35  6384.3  872.16
#Mann=5,-1,0
  4535.2    0.05       0  4842.8    0.12       0  4988.2    0.07       0
  5007.0    0.12       0  5085.8    0.05       0
Bank Sta=4988.2,5007
Exp/Cntr=0.3,0.1

Type RM Length L Ch R = 1,48731,285,285,285
BEGIN DESCRIPTION:
Mapping XS 2ac60920
END DESCRIPTION:
XS GIS Cut Line= 2
      2260771.30      7145612.19      2260804.54      7143378.14
#Sta/Elev= 30
  4455.3  874.49  4577.5  866.86  4697.5  863.02  4726.6  863.26  4757.5  862.76
  4797.5  860.63  4867.5  859.74  4907.5  857.81  4917.5  856.23  4977.5  856.37
  4997.5  853.95  5017.6  848.10  5018.2  844.15  5020.2  843.65  5037.0  844.15
  5037.6  845.66  5047.6  850.16  5055.4  852.63  5077.6  859.63  5087.6  860.00
  5147.6  858.88  5167.6  859.45  5397.6  858.11  5677.6  857.70  5777.6  858.39
  5797.6  857.80  6397.7  862.27  6597.7  865.93  6677.7  870.09  6689.6  869.98
#Mann=5,-1,0
  4455.3    0.05       0  4726.6    0.12       0  5018.2    0.07       0
  5037.0    0.12       0  5055.4    0.05       0
Bank Sta=5018.2,5037
Exp/Cntr=0.3,0.1

Type RM Length L Ch R = 1,48446,483,483,483
BEGIN DESCRIPTION:
Catlett Creek 46.0
END DESCRIPTION:
XS GIS Cut Line= 3
      2261029.00      7145559.98      2261018.49      7145158.82
      2261219.31      7143954.34
#Sta/Elev= 30
  4598.7  872.06  4920.3  858.99  4958.8  858.95  4968.8  857.78  4978.8  850.02
  4979.4  842.57  4981.4  842.07  4998.2  842.57  5008.9  845.31  5028.8  853.38
  5033.9  851.15  5039.4  853.81  5049.5  856.29  5110.3  853.68  5142.0  853.50
  5171.1  853.28  5242.1  858.42  5277.2  857.52  5485.4  858.88  5505.7  857.49
  5536.1  858.66  5576.2  857.31  5617.2  858.72  5627.4  857.14  5688.2  857.51
  5702.9  856.48  5885.3  858.09  6093.7  862.00  6189.4  867.16  6221.1  866.88
#Mann=5,-1,0
  4598.7    0.05       0  4920.3    0.12       0  4979.4    0.07       0
  4998.2    0.12       0  5142.0    0.05       0
Bank Sta=4979.4,4998.2
Exp/Cntr=0.3,0.1

Type RM Length L Ch R = 1,47963,502,502,502
BEGIN DESCRIPTION:
Catlett Creek 45.0
END DESCRIPTION:
XS GIS Cut Line= 3
      2261442.14      7145668.43      2261419.70      7145099.57
      2261541.96      7144160.20
#Sta/Elev= 30
  4430.7  876.73  4749.4  861.90  4789.4  857.22  4899.5  856.83  4919.5  859.44
  4933.7  859.17  4969.5  853.89  4979.6  849.02  4987.9  840.69  4989.9  840.19
  5006.7  840.69  5019.7  847.04  5034.1  846.88  5060.1  854.47  5071.7  855.28
  5090.3  857.01  5231.5  857.74  5463.5  855.51  5604.6  857.26  5624.8  856.94
  5634.9  854.46  5651.6  856.68  5695.4  856.73  5735.7  864.14  5766.0  861.19
  5786.1  862.74  5804.7  866.73  5858.1  871.49  5897.1  880.66  5947.3  880.62
#Mann=7,-1,0
  4430.7    0.05       0  4933.7    0.12       0  4987.9    0.07       0
  5006.7    0.12       0  5071.7    0.05       0  5463.5    0.12       0
  5858.1    0.05       0
Bank Sta=4987.9,5006.7
Exp/Cntr=0.3,0.1

Type RM Length L Ch R = 1,47461,718,718,718
BEGIN DESCRIPTION:
Catlett Creek 44.0
END DESCRIPTION:
XS GIS Cut Line= 3
      2262059.69      7145356.76      2261885.21      7145052.20
      2261757.62      7144324.60
#Sta/Elev= 30
  4649.0  875.18  4698.9  869.60  4806.8  861.92  4860.0  860.80  4897.8  858.16
  4940.6  855.37  4956.4  852.10  4978.0  845.21  4981.6  840.70  4983.6  840.20
  5000.5  840.70  5007.2  841.87  5012.4  849.26  5022.5  854.06  5032.7  855.72
  5066.6  853.45  5144.6  854.71  5192.3  855.32  5225.6  854.43  5407.8  855.29
  5412.9  851.89  5467.2  858.15  5472.3  855.52  5479.4  856.70  5511.1  856.73
  5550.5  857.37  5580.9  860.41  5591.1  863.06  5640.3  868.99  5738.7  873.75
#Mann=7,-1,0
  4649.0    0.05       0  4897.8    0.12       0  4981.6    0.07       0
  5000.5    0.12       0  5144.6    0.05       0  5192.3    0.12       0
  5511.1    0.05       0
Bank Sta=4981.6,5000.5
Exp/Cntr=0.3,0.1

Type RM Length L Ch R = 1,46743,776,776,776
BEGIN DESCRIPTION:
Catlett Creek 43.0
END DESCRIPTION:
XS GIS Cut Line= 3
      2262501.57      7145122.68      2262380.00      7144737.14
      2262092.98      7144053.60
#Sta/Elev= 30
  4610.9  868.45  4665.1  866.89  4687.1  864.99  4702.7  865.46  4735.1  862.62
  4767.4  861.93  4812.9  858.28  4832.1  858.54  4837.4  857.34  4874.0  855.60
  4949.2  854.79  4959.7  851.81  4966.8  845.07  4989.6  838.15  4991.6  837.65
  5008.6  838.15  5011.0  844.11  5015.2  844.11  5029.5  852.46  5058.7  851.33
  5077.0  854.03  5129.9  853.75  5164.6  851.70  5188.0  852.60  5336.3  853.24
  5442.2  855.45  5511.0  858.85  5624.8  867.67  5695.3  871.41  5756.5  877.00
#Mann=5,-1,0
  4610.9    0.05       0  4874.0    0.12       0  4989.6    0.07       0
  5008.6    0.12       0  5188.0    0.05       0
Bank Sta=4989.6,5008.6
Exp/Cntr=0.3,0.1

Type RM Length L Ch R = 1,45967,404,404,404
BEGIN DESCRIPTION:
Catlett Creek 42.0
END DESCRIPTION:
XS GIS Cut Line= 3
      2262934.99      7145126.60      2262737.18      7144172.47
      2262708.82      7143793.15
#Sta/Elev= 30
  4013.1  864.58  4030.1  862.88  4101.5  859.64  4224.1  855.24  4244.5  855.92
  4262.1  853.83  4346.6  851.65  4530.5  851.68  4602.0  852.77  4858.9  850.58
  4898.1  851.13  4904.0  851.98  4949.0  851.92  4959.4  851.10  4969.6  848.63
  4986.2  840.25  4990.5  836.57  4992.5  836.07  5009.5  836.57  5032.7  851.73
  5110.3  854.95  5150.4  858.37  5159.9  860.87  5170.5  861.44  5180.5  863.95
  5210.6  863.36  5280.8  868.66  5290.8  868.66  5330.9  873.62  5367.9  875.57
#Mann=3,-1,0
  4013.1     0.1       0  4990.5    0.07       0  5009.5    0.05       0
#XS Ineff=2,0
    0.00 4609.50  864.54               0
Permanent Ineff=
       F       F
Bank Sta=4990.5,5009.5
Exp/Cntr=0.3,0.1

Type RM Length L Ch R = 1,45563,319,319,319
BEGIN DESCRIPTION:
Catlett Creek 41.0
END DESCRIPTION:
XS GIS Cut Line= 3
      2263159.23      7145100.94      2263121.46      7144144.83
      2263098.27      7143819.11
#Sta/Elev= 30
  4058.7  869.68  4079.7  869.62  4129.7  866.09  4169.7  860.81  4188.0  862.14
  4209.8  859.28  4278.4  855.26  4319.8  852.73  4419.9  850.91  4560.0  851.80
  4600.1  850.70  4630.1  851.56  4960.3  849.25  4970.3  848.79  4980.4  843.94
  5000.4  839.14  5000.9  836.00  5002.9  835.50  5019.9  836.00  5020.5  837.57
  5030.4  843.04  5040.4  850.58  5123.1  853.90  5130.7  855.63  5170.8  857.70
  5220.9  863.71  5241.0  863.60  5258.7  866.02  5263.7  865.24  5342.1  873.91
#Mann=4,-1,0
  4058.7    0.12       0  4278.4     0.1       0  5000.9    0.03       0
  5019.9    0.05       0
#XS Ineff=2,0
    0.00 4750.00  861.89               0
Permanent Ineff=
       F       F
Bank Sta=5000.9,5019.9
Exp/Cntr=0.3,0.1

Type RM Length L Ch R = 1,45244,72,72,72
BEGIN DESCRIPTION:
Catlett Creek 40.0
END DESCRIPTION:
XS GIS Cut Line= 3
      2263502.97      7145081.57      2263409.09      7144200.60
      2263161.07      7143827.22
#Sta/Elev= 30
  4158.0  878.09  4166.6  877.07  4310.4  862.27  4407.2  855.95  4451.2  853.11
  4521.2  852.75  4551.8  850.79  4618.6  850.10  4692.6  852.15  4711.1  849.74
  4732.8  849.42  4944.0  849.09  4983.9  835.26  4985.9  834.76  5003.0  835.26
  5034.5  846.75  5047.3  847.96  5051.9  850.98  5057.9  848.93  5067.0  850.10
  5073.0  849.14  5088.0  852.09  5094.0  850.75  5103.0  852.69  5175.2  856.09
  5181.2  855.15  5238.3  860.82  5340.6  864.77  5484.9  867.23  5492.2  868.49
#Mann=5,-1,0
  4158.0    0.05       0  4166.6    0.12       0  4407.2    0.04       0
  4983.9    0.05       0  5003.0    0.05       0
#XS Ineff=2,0
    0.00 4831.90  864.69               0
Permanent Ineff=
       F       F
Bank Sta=4983.9,5003
Exp/Cntr=0.3,0.1

Type RM Length L Ch R = 1,45172,462,462,462
BEGIN DESCRIPTION:
Catlett Creek 39.5
END DESCRIPTION:
XS GIS Cut Line= 3
      2263660.13      7145024.55      2263458.73      7144149.03
      2263205.13      7143837.36
#Sta/Elev= 30
  4205.0  873.73  4289.4  866.48  4324.6  862.71  4421.0  856.32  4507.2  850.99
  4835.6  848.71  4907.4  849.86  4938.2  844.73  4944.7  842.34  4949.8  844.70
  4979.3  839.22  4990.2  835.11  4992.2  834.61  5009.3  835.11  5010.0  837.28
  5020.3  839.09  5061.3  842.98  5083.4  847.20  5130.6  848.81  5138.5  850.99
  5159.3  851.19  5173.7  853.88  5194.5  854.26  5258.4  860.02  5295.0  859.68
  5365.4  863.82  5443.7  865.05  5450.2  863.47  5478.9  866.06  5505.2  865.70
#Mann=5,-1,0
  4205.0    0.05       0  4289.4    0.12       0  4421.0    0.05       0
  4990.2    0.04       0  5009.3    0.05       0
#XS Ineff=2,0
    0.00 4877.30  863.10               0
Permanent Ineff=
       F       F
Bank Sta=4990.2,5009.3
Exp/Cntr=0.3,0.1

Type RM Length L Ch R = 1,44710,627,627,627
BEGIN DESCRIPTION:
Catlett Creek 39.0
END DESCRIPTION:
XS GIS Cut Line= 3
      2264588.58      7144240.08      2263812.41      7143976.52
      2263209.26      7143822.10
#Sta/Elev= 30
  4180.3  874.80  4201.2  876.81  4232.7  871.41  4274.9  871.38  4296.0  868.00
  4319.8  867.91  4521.9  857.52  4635.4  851.41  4834.6  846.76  4950.8  847.22
  4961.4  846.21  4970.1  840.76  4975.4  840.60  4983.5  832.49  4985.5  831.99
  5002.6  832.49  5048.2  839.38  5065.5  844.93  5089.0  843.25  5096.4  846.88
  5293.0  848.30  5369.5  851.94  5395.8  855.62  5451.1  857.32  5478.4  860.61
  5499.0  858.51  5540.3  862.36  5550.6  859.91  5568.3  863.81  5622.6  865.76
#Mann=5,-1,0
  4180.3    0.05       0  4319.8    0.12       0  4521.9    0.05       0
  4983.5    0.04       0  5002.6    0.05       0
#XS Ineff=2,0
    0.00 4859.60  861.19 5140.40    0.00  861.19
Permanent Ineff=
       F       F
Bank Sta=4983.5,5002.6
Exp/Cntr=0.3,0.1

Type RM Length L Ch R = 1,44083,521,521,521
BEGIN DESCRIPTION:
Catlett Creek 38.0
END DESCRIPTION:
XS GIS Cut Line= 3
      2264594.65      7143667.16      2263838.30      7143386.08
      2263075.07      7143496.81
#Sta/Elev= 30
  4183.9  884.40  4232.6  883.37  4273.8  878.84  4296.6  875.63  4303.4  873.32
  4333.8  870.67  4371.3  864.10  4488.6  854.63  4519.6  851.02  4560.6  848.28
  4691.3  845.32  4872.7  844.53  4979.4  846.25  4987.7  843.39  4993.0  843.39
  5010.8  831.53  5012.8  831.03  5029.9  831.53  5030.5  835.33  5049.3  842.97
  5054.3  842.88  5060.8  845.55  5070.9  846.69  5101.2  845.48  5273.0  847.02
  5576.1  851.47  5610.8  852.25  5626.7  853.95  5667.1  853.40  5762.0  855.30
#Mann=5,-1,0
  4183.9    0.05       0  4273.8    0.12       0  4519.6    0.05       0
  5010.8    0.04       0  5029.9    0.05       0
#XS Ineff=2,0
    0.00 4868.00  863.71 5132.00    0.00  863.71
Permanent Ineff=
       F       F
Bank Sta=5010.8,5029.9
Exp/Cntr=0.3,0.1

Type RM Length L Ch R = 1,43562,479,479,479
BEGIN DESCRIPTION:
Catlett Creek 37.0
END DESCRIPTION:
XS GIS Cut Line= 3
      2264629.03      7143660.03      2263879.00      7142910.00
      2263179.01      7142710.00
#Sta/Elev= 30
  3939.3  885.74  4052.3  879.10  4109.0  872.78  4193.9  866.18  4349.5  861.00
  4424.5  852.31  4434.3  850.91  4476.7  855.40  4519.2  845.05  4561.6  846.43
  4618.2  844.23  4787.9  843.02  4929.3  844.33  4943.4  841.41  4957.6  834.87
  4961.8  830.92  4963.8  830.42  4981.6  830.92  5002.6  834.01  5016.9  845.06
  5055.9  843.22  5072.8  845.18  5156.0  844.82  5176.8  846.91  5260.0  845.74
  5499.2  847.67  5592.8  854.93  5644.8  863.92  5686.4  868.23  5728.0  869.48
#Mann=5,-1,0
  3939.3    0.05       0  4052.3    0.12       0  4424.5    0.05       0
  4961.8    0.04       0  4981.6    0.05       0
#XS Ineff=2,0
       0                 5160.60    0.00  862.63
Permanent Ineff=
       F       F
Bank Sta=4961.8,4981.6
Exp/Cntr=0.3,0.1

Type RM Length L Ch R = 1,43083,658,658,658
BEGIN DESCRIPTION:
Catlett Creek 36.0
END DESCRIPTION:
XS GIS Cut Line= 3
      2264571.95      7143429.81      2264062.45      7142526.95
      2263713.31      7141981.29
#Sta/Elev= 30
  3963.3  870.49  4098.3  862.56  4163.3  860.31  4341.0  848.92  4384.3  847.00
  4399.4  847.54  4443.5  844.37  4508.5  841.83  4560.2  843.36  4627.0  841.58
  4713.6  842.94  4751.2  841.49  4794.5  843.00  4918.7  842.33  4934.6  840.79
  4972.1  841.71  4977.9  841.47  4985.0  838.63  4988.3  829.57  4990.3  829.07
  5008.6  829.57  5030.1  834.50  5057.2  843.71  5102.9  842.59  5170.2  843.84
  5327.0  845.45  5332.9  846.54  5390.4  846.81  5463.1  849.10  5647.8  861.35
#Mann=4,-1,0
  3963.3    0.05       0  4988.3    0.07       0  5008.6    0.05       0
  5170.2    0.05       0
Bank Sta=4988.3,5008.6
Exp/Cntr=0.3,0.1

Type RM Length L Ch R = 1,42425,450,450,450
BEGIN DESCRIPTION:
Catlett Creek 35.0
END DESCRIPTION:
XS GIS Cut Line= 3
      2264873.60      7143230.15      2264529.00      7142260.00
      2264097.69      7141699.72
#Sta/Elev= 30
  3970.5  866.10  3998.2  861.30  4090.8  856.90  4178.0  848.16  4263.3  843.63
  4743.1  838.35  4923.4  839.98  4953.8  836.58  4959.1  838.21  4984.6  831.34
  4989.9  832.84  4997.4  828.61  5003.2  828.61  5003.4  824.86  5005.4  824.36
  5023.8  824.86  5028.1  825.04  5036.3  830.39  5042.6  828.09  5057.1  840.04
  5063.4  837.44  5071.6  840.58  5090.1  841.25  5291.8  843.62  5470.3  852.22
  5514.9  857.20  5555.4  860.54  5628.0  860.87  5642.5  864.04  5707.1  866.86
#Mann=7,-1,0
  3970.5    0.12       0  4263.3    0.05       0  4923.4    0.12       0
  5003.4    0.07       0  5023.8    0.12       0  5090.1    0.05       0
  5514.9    0.12       0
Bank Sta=5003.4,5023.8
Exp/Cntr=0.3,0.1

Type RM Length L Ch R = 1,41975,590,590,590
BEGIN DESCRIPTION:
Catlett Creek 34.0
END DESCRIPTION:
XS GIS Cut Line= 3
      2265203.45      7143085.80      2264927.98      7142193.98
      2264633.02      7141523.27
#Sta/Elev= 30
  4066.6  857.89  4098.7  857.28  4145.9  851.92  4169.2  852.23  4206.6  848.99
  4234.5  849.08  4240.1  846.68  4268.6  845.24  4365.1  840.80  4784.4  836.80
  4959.1  840.07  4972.8  840.87  4984.0  833.59  4989.3  823.79  4991.3  823.29
  5009.7  823.79  5009.8  826.69  5038.6  835.96  5056.5  834.71  5062.0  836.06
  5079.9  832.98  5091.7  834.54  5102.7  839.27  5155.4  841.10  5190.1  838.85
  5245.3  840.58  5410.7  843.80  5626.2  858.87  5648.9  858.99  5732.7  867.84
#Mann=7,-1,0
  4066.6    0.05       0  4206.6    0.12       0  4268.6    0.05       0
  4959.1    0.12       0  4989.3    0.07       0  5009.7    0.12       0
  5245.3    0.05       0
Bank Sta=4989.3,5009.7
Exp/Cntr=0.3,0.1

Type RM Length L Ch R = 1,41385,550,550,550
BEGIN DESCRIPTION:
Catlett Creek 33.0
END DESCRIPTION:
XS GIS Cut Line= 3
      2265474.27      7143028.46      2265212.71      7141826.59
      2264931.90      7141364.41
#Sta/Elev= 30
  3770.0  859.24  3821.5  854.95  3850.3  847.17  3860.4  846.55  3865.5  843.69
  3881.0  842.80  3914.6  842.78  3932.2  849.09  3942.4  849.13  4056.8  841.18
  4177.8  838.24  4536.0  836.01  4863.5  837.78  4894.2  839.66  4917.8  837.04
  4935.1  834.70  4948.7  836.83  4965.8  831.29  4976.0  830.66  4986.3  824.78
  4986.8  820.43  4988.8  819.93  5007.2  820.43  5007.7  825.44  5015.2  833.60
  5030.7  838.57  5232.3  837.40  5342.7  842.22  5459.0  851.38  5540.8  863.32
#Mann=4,-1,0
  3770.0    0.05       0  4917.8    0.12       0  4986.8    0.07       0
  5007.2    0.12       0
Bank Sta=4986.8,5007.2
Exp/Cntr=0.3,0.1

Type RM Length L Ch R = 1,40835,579,579,579
BEGIN DESCRIPTION:
Catlett Creek 32.0
END DESCRIPTION:
XS GIS Cut Line= 3
      2265604.49      7143045.85      2265679.00      7141960.00
      2265522.20      7140995.47
#Sta/Elev= 30
  3911.5  865.81  4017.6  856.02  4046.6  851.78  4051.6  852.48  4077.7  848.34
  4117.8  846.61  4208.0  846.22  4268.2  838.66  4378.4  836.65  4408.5  837.71
  4634.4  835.69  4649.1  836.82  4679.2  835.22  4899.7  835.93  4930.8  836.47
  4939.8  837.79  4959.8  833.69  4967.1  830.16  4979.9  826.54  4987.2  819.25
  4989.2  818.75  5007.6  819.25  5028.1  837.03  5033.2  835.87  5040.4  837.64
  5073.5  835.88  5212.7  835.94  5273.4  837.52  5425.4  838.16  5977.1  845.03
#Mann=5,-1,0
  3911.5    0.05       0  4967.1    0.12       0  4987.2    0.07       0
  5007.6    0.12       0  5073.5    0.05       0
Bank Sta=4987.2,5007.6
Exp/Cntr=0.3,0.1

Type RM Length L Ch R = 1,40256,542,542,542
BEGIN DESCRIPTION:
Catlett Creek 31.0
END DESCRIPTION:
XS GIS Cut Line= 3
      2266128.29      7143096.19      2266179.00      7142160.00
      2266701.71      7141247.24
#Sta/Elev= 30
  4061.5  853.57  4147.8  847.45  4157.8  844.77  4170.0  845.48  4288.0  839.93
  4535.1  835.46  4808.8  834.95  4858.9  833.48  4905.3  835.52  4949.0  834.19
  4963.6  828.00  4979.0  824.01  4986.0  818.26  4988.1  817.76  5007.2  818.26
  5012.7  824.27  5028.6  834.93  5141.4  833.90  5183.4  833.15  5211.3  830.76
  5218.0  832.65  5241.1  834.32  5254.5  833.15  5313.5  834.01  5344.8  830.94
  5366.7  833.61  5549.4  835.30  5698.3  842.72  5784.8  846.96  6050.9  865.10
#Mann=7,-1,0
  4061.5    0.05       0  4963.6    0.12       0  4986.0    0.07       0
  5007.2    0.12       0  5141.4    0.05       0  5698.3    0.12       0
  5784.8    0.05       0
Bank Sta=4986,5007.2
Exp/Cntr=0.3,0.1

Type RM Length L Ch R = 1,39714,1278,1278,1278
BEGIN DESCRIPTION:
Catlett Creek 30.0
END DESCRIPTION:
XS GIS Cut Line= 3
      2266472.55      7143089.22      2266640.51      7142159.67
      2266769.64      7141299.51
#Sta/Elev= 30
  4055.4  850.89  4178.8  840.22  4186.7  841.34  4207.0  841.09  4257.8  837.91
  4481.4  832.90  4755.8  832.05  4867.6  832.85  4917.2  834.77  4938.7  834.49
  4948.9  831.94  4958.7  827.68  4963.7  827.88  4969.2  825.49  4978.9  817.03
  4981.0  816.53  5000.2  817.03  5009.8  823.40  5019.2  831.97  5024.2  832.47
  5050.2  829.76  5084.1  831.37  5201.9  832.81  5414.3  838.56  5515.4  843.48
  5586.7  845.58  5590.2  845.82  5687.3  852.80  5699.8  852.53  5869.8  862.55
#Mann=7,-1,0
  4055.4    0.05       0  4917.2    0.12       0  4978.9    0.07       0
  5000.2    0.12       0  5084.1    0.05       0  5586.7    0.12       0
  5590.2    0.05       0
Bank Sta=4978.9,5000.2
Exp/Cntr=0.3,0.1

Type RM Length L Ch R = 1,38436,664,664,664
BEGIN DESCRIPTION:
Catlett Creek 29.0
END DESCRIPTION:
XS GIS Cut Line= 3
      2266763.24      7143647.52      2267712.45      7142470.28
      2268222.36      7141609.29
#Sta/Elev= 30
  3431.5  852.76  3518.5  848.16  3590.5  846.98  3660.9  843.15  3683.2  843.51
  3732.8  838.01  3753.6  837.58  3775.1  839.40  3803.2  833.63  3896.0  830.39
  3995.1  829.54  4379.0  830.81  4735.6  828.82  4953.9  831.27  4969.8  829.21
  4985.4  821.03  5001.0  818.03  5003.0  815.13  5005.2  814.63  5024.7  815.13
  5028.3  820.25  5037.0  823.81  5049.7  832.24  5080.9  830.69  5139.4  832.20
  5145.2  831.37  5374.4  837.92  5533.2  841.98  5751.6  844.33  5944.4  849.40
#Mann=5,-1,0
  3431.5    0.05       0  4953.9    0.12       0  5003.0    0.07       0
  5024.7    0.12       0  5374.4    0.05       0
Bank Sta=5003,5024.7
Exp/Cntr=0.3,0.1

Type RM Length L Ch R = 1,37772,685,685,685
BEGIN DESCRIPTION:
Catlett Creek 28.5
END DESCRIPTION:
XS GIS Cut Line= 3
      2268064.46      7143720.26      2268069.72      7142848.77
      2268206.44      7141756.29
#Sta/Elev= 30
  4128.5  847.13  4198.8  842.57  4258.8  834.41  4408.8  827.03  4438.8  814.17
  4458.8  827.94  4501.6  828.99  4578.8  827.91  4648.8  830.04  4678.8  827.39
  4728.8  827.31  4798.8  828.25  4808.8  830.24  4838.8  828.17  4927.7  828.39
  4948.8  828.95  4968.8  817.27  4978.8  817.32  4986.0  812.81  4988.2  812.31
  5007.7  812.81  5018.9  821.65  5034.2  829.98  5068.2  828.39  5291.0  828.32
  5517.7  832.63  5532.9  834.55  5563.1  833.62  5920.6  839.96  6101.0  844.71
#Mann=6,-1,0
  4128.5    0.12       0  4501.6    0.05       0  4927.7    0.12       0
  4986.0    0.07       0  5007.7    0.12       0  5068.2    0.05       0
Bank Sta=4986,5007.7
Exp/Cntr=0.3,0.1

Type RM Length L Ch R = 1,37087,660,660,660
BEGIN DESCRIPTION:
Catlett Creek 28.0
END DESCRIPTION:
XS GIS Cut Line= 3
      2268673.66      7144055.31      2268654.19      7143010.49
      2268762.19      7141664.82
#Sta/Elev= 30
  3955.0  862.02  3990.3  863.68  4010.3  856.93  4080.3  850.25  4240.4  842.82
  4280.4  837.83  4330.4  836.97  4430.4  829.80  4790.5  822.72  4953.6  826.36
  4960.5  825.61  4968.0  809.69  4970.5  809.19  4993.0  809.69  5010.5  814.04
  5030.6  826.44  5040.6  827.23  5140.9  826.96  5181.1  821.21  5201.1  825.95
  5262.1  825.10  5374.7  824.68  5391.7  828.30  5431.9  825.99  5625.1  826.94
  5863.3  831.50  6243.5  848.58  6284.6  851.67  6334.8  859.22  6350.0  858.10
#Mann=5,-1,0
  3955.0    0.05       0  4953.6    0.12       0  4968.0    0.07       0
  4993.0    0.12       0  5262.1    0.05       0
Bank Sta=4968,4993
Exp/Cntr=0.3,0.1

Type RM Length L Ch R = 1,36427,1096,1096,1096
BEGIN DESCRIPTION:
Catlett Creek 27.0
END DESCRIPTION:
XS GIS Cut Line= 3
      2269029.00      7144210.03      2268979.00      7142660.00
      2268898.25      7141683.27
#Sta/Elev= 30
  3449.5  869.51  3569.6  863.89  3629.6  857.57  3659.6  856.98  3689.7  853.33
  3839.7  844.28  3909.8  837.50  4109.9  826.37  4350.0  821.62  4470.1  824.29
  4883.3  824.68  4940.3  825.17  4977.8  807.92  4980.3  807.42  5002.8  807.92
  5010.4  812.54  5040.5  816.90  5063.3  823.53  5080.6  822.02  5120.7  825.71
  5168.3  824.94  5281.3  828.10  5305.1  827.51  5426.0  831.70  5783.0  850.11
  5863.3  856.57  5883.3  859.57  5914.5  857.58  5963.6  859.23  5980.4  861.27
#Mann=5,-1,0
  3449.5    0.05       0  4883.3    0.12       0  4977.8    0.07       0
  5002.8    0.12       0  5168.3    0.05       0
Bank Sta=4977.8,5002.8
Exp/Cntr=0.3,0.1

Type RM Length L Ch R = 1,35331,533,533,533
BEGIN DESCRIPTION:
Catlett Creek 26.0
END DESCRIPTION:
XS GIS Cut Line= 3
      2269179.00      7144160.02      2269429.00      7142610.00
      2269479.00      7142209.97
#Sta/Elev= 30
  3429.2  867.67  3550.8  864.60  3631.8  859.03  3763.5  845.54  4118.0  823.19
  4249.7  820.49  4342.9  823.43  4697.6  823.67  4877.7  824.61  4904.0  820.55
  4909.1  824.07  4918.2  823.37  4958.7  807.80  4965.8  806.70  4970.9  808.95
  4976.6  806.24  4979.1  805.74  5001.6  806.24  5009.3  808.36  5019.4  816.64
  5037.0  818.09  5042.1  812.98  5049.6  815.85  5059.7  815.57  5079.9  824.24
  5097.4  823.83  5150.4  822.99  5221.0  827.61  5261.3  833.81  5402.4  845.60
#Mann=5,-1,0
  3429.2    0.05       0  4697.6    0.12       0  4976.6    0.07       0
  5001.6    0.12       0  5097.4    0.05       0
Bank Sta=4976.6,5001.6
Exp/Cntr=0.3,0.1

Type RM Length L Ch R = 1,34798,600,600,600
BEGIN DESCRIPTION:
Catlett Creek 25.0
END DESCRIPTION:
XS GIS Cut Line= 3
      2269329.00      7144010.01      2269879.00      7142460.00
      2269929.00      7142060.01
#Sta/Elev= 30
  3354.4  860.56  3426.3  858.39  3431.6  856.53  3488.0  853.71  3493.3  856.06
  3524.2  853.53  3544.4  848.90  3549.7  850.05  3556.0  848.17  3724.3  834.65
  3729.7  835.73  3760.5  833.60  3778.8  829.19  3873.4  824.16  4044.1  821.82
  4089.5  819.40  4233.2  822.54  4685.1  822.21  4882.4  823.20  4946.0  821.67
  4983.7  807.96  4983.9  804.79  4986.4  804.29  5008.9  804.79  5029.3  823.92
  5140.2  827.43  5220.8  832.11  5278.8  838.21  5321.6  839.38  5402.2  850.17
#Mann=4,-1,0
  3354.4    0.05       0  4685.1    0.12       0  4983.9    0.07       0
  5008.9    0.12       0
Bank Sta=4983.9,5008.9
Exp/Cntr=0.3,0.1

Type RM Length L Ch R = 1,34198,662,662,662
BEGIN DESCRIPTION:
Catlett Creek 24.5
END DESCRIPTION:
XS GIS Cut Line= 3
      2269434.84      7143898.27      2270152.27      7142933.36
      2270132.64      7142043.78
#Sta/Elev= 30
  3797.6  856.89  3849.0  849.27  3857.4  850.23  3913.7  843.48  3928.3  843.80
  3993.0  837.71  4063.9  829.00  4113.9  826.51  4449.7  822.15  4892.6  819.87
  4950.4  820.01  4965.0  816.34  4979.3  807.67  4979.5  803.23  4982.0  802.73
  5004.5  803.23  5023.4  803.52  5063.4  812.86  5083.4  813.60  5103.4  821.33
  5113.4  823.11  5163.4  822.87  5173.4  819.80  5183.4  813.34  5193.4  819.11
  5233.4  822.27  5443.5  821.70  5648.6  826.26  5803.6  836.91  5889.8  844.96
#Mann=5,-1,0
  3797.6    0.05       0  4892.6    0.12       0  4979.5    0.07       0
  5004.5    0.12       0  5648.6    0.05       0
Bank Sta=4979.5,5004.5
Exp/Cntr=0.3,0.1

Type RM Length L Ch R = 1,33536,531,531,531
BEGIN DESCRIPTION:
Catlett Creek 24.0
END DESCRIPTION:
XS GIS Cut Line= 3
      2270393.70      7144304.78      2270594.18      7143309.57
      2270828.63      7142103.14
#Sta/Elev= 30
  3984.8  835.33  4203.9  832.00  4290.4  829.33  4341.2  825.73  4346.7  823.86
  4386.9  826.15  4499.7  820.60  4662.9  818.94  4907.8  821.50  4938.4  818.17
  4951.1  812.85  4969.0  810.23  4976.9  802.15  4979.4  801.65  5001.9  802.15
  5002.3  803.99  5019.9  818.41  5030.1  822.26  5048.5  823.63  5070.9  819.94
  5092.2  820.02  5508.9  818.70  5787.2  823.06  5936.8  832.53  5987.7  836.56
  6008.1  840.13  6038.6  841.85  6045.6  843.46  6059.0  842.96  6229.0  851.24
#Mann=4,-1,0
  3984.8    0.12       0  4976.9    0.07       0  5001.9    0.12       0
  5092.2    0.05       0
Bank Sta=4976.9,5001.9
Exp/Cntr=0.3,0.1

Type RM Length L Ch R = 1,33005,328,328,328
BEGIN DESCRIPTION:
Catlett Creek 23.5
END DESCRIPTION:
XS GIS Cut Line= 3
      2270951.71      7144517.89      2271040.77      7143557.70
      2270827.50      7142293.37
#Sta/Elev= 30
  3995.0  841.49  4043.1  836.42  4173.7  827.25  4273.9  822.27  4444.8  818.12
  4595.5  817.53  4655.7  814.61  4685.8  817.55  4836.5  817.53  4906.8  819.43
  4947.0  817.23  4959.3  813.57  4964.8  801.16  4967.3  800.66  4989.8  801.16
  5001.3  802.04  5028.0  818.40  5038.1  819.82  5078.7  819.36  5088.8  820.75
  5118.7  818.16  5251.1  819.97  5359.1  817.35  5494.5  819.44  5808.8  818.33
  5869.7  819.75  5972.1  825.94  6079.9  834.68  6110.6  834.28  6241.5  843.60
#Mann=7,-1,0
  3995.0    0.05       0  4273.9    0.12       0  4964.8    0.07       0
  4989.8    0.12       0  5118.7    0.05       0  5972.1    0.12       0
  6110.6    0.05       0
Bank Sta=4964.8,4989.8
Exp/Cntr=0.3,0.1

Type RM Length L Ch R = 1,32677,749,749,749
BEGIN DESCRIPTION:
Catlett Creek 23.0
END DESCRIPTION:
XS GIS Cut Line= 3
      2272047.83      7143767.24      2271315.61      7143573.54
      2270883.15      7142373.48
#Sta/Elev= 30
  4242.6  834.83  4430.1  823.66  4490.2  820.97  4600.8  817.73  4710.4  817.51
  4934.4  818.87  4944.8  817.72  4957.7  810.24  4975.8  805.37  4980.3  799.74
  4982.8  799.24  5005.3  799.74  5006.9  803.24  5014.4  809.14  5037.6  814.82
  5147.0  817.80  5890.3  817.72  5921.2  816.69  5971.0  819.85  6002.6  829.33
  6033.3  832.57  6038.6  830.57  6077.3  837.48  6094.7  838.43  6100.0  836.53
  6109.2  837.55  6130.7  834.34  6156.1  833.80  6194.3  840.00  6275.6  840.89
#Mann=8,-1,0
  4242.6    0.05       0  4430.1    0.12       0  4490.2    0.05       0
  4710.4    0.12       0  4980.3    0.07       0  5005.3    0.12       0
  5147.0    0.05       0  5890.3    0.12       0
Bank Sta=4980.3,5005.3
Exp/Cntr=0.3,0.1

Type RM Length L Ch R = 1,31928,409,409,409
BEGIN DESCRIPTION:
Catlett Creek 22.0
END DESCRIPTION:
XS GIS Cut Line= 3
      2272128.99      7143259.99      2271738.81      7143099.49
      2270978.98      7142509.98
#Sta/Elev= 30
  4578.1  842.55  4767.3  829.53  4830.0  825.30  4877.9  818.02  4936.6  816.74
  4977.5  799.65  4980.0  799.15  5002.5  799.65  5021.2  804.89  5035.7  810.91
  5042.0  816.33  5063.0  818.65  5106.3  815.79  5191.4  815.88  5214.0  817.45
  5245.3  815.57  5334.4  816.93  5355.2  819.12  5384.2  816.59  5442.1  815.73
  5462.9  817.67  5626.8  816.76  5676.5  817.63  5691.0  819.58  5711.8  817.49
  5733.8  817.76  5770.6  820.48  5904.6  830.97  5933.6  837.93  5961.7  841.44
#Mann=6,-1,0
  4578.1    0.05       0  4767.3    0.12       0  4977.5    0.07       0
  5002.5    0.12       0  5245.3    0.05       0  5770.6    0.12       0
Bank Sta=4977.5,5002.5
Exp/Cntr=0.3,0.1
