--- Denton Creek Tributary 17.prj (project) ---

Proj Title=Denton Creek Tributary 17 Base Level Engineering
Current Plan=p01
Default Exp/Contr=0.3,0.1
English Units
Geom File=g01
Flow File=f01
Plan File=p01
Y Axis Title=Elevation
X Axis Title(PF)=Main Channel Distance
X Axis Title(XS)=Station
BEGIN DESCRIPTION:
Denton Creek Tributary 17
END DESCRIPTION:
DSS Export Rating Curves= 0
DSS Export Rating Curve Sorted= 0
DSS Export Volume Flow Curves= 0
DXF OffsetX= 0
DXF OffsetY= 0
DXF ScaleX= 1
DXF ScaleY= 10

--- Denton Creek Tributary 17.p01 (plan) ---

Plan Title=Multiple Run
Short Identifier=Multiple
Geom File=g01
Flow File=f01
Subcritical Flow
K Sum by GR= 0
Std Step Tol= 0.01
Critical Tol= 0.01
Num of Std Step Trials= 20
Max Error Tol= 0.3
Flow Tol Ratio= 0.001
Split Flow NTrial= 30
Split Flow Tol= 0.02
Split Flow Ratio= 0.02
Log Output Level= 0
Friction Slope Method= 1
Unsteady Friction Slope Method= 2
Unsteady Bridges Friction Slope Method= 1
Parabolic Critical Depth
Global Vel Dist=  1 , 1 , 1
Global Log Level= 0
CheckData=True
Encroach Param= -1, 0, 0, 0
BEGIN DESCRIPTION:
Multiple Run
END DESCRIPTION:

--- Denton Creek Tributary 17.f01 (steady flow) ---

Flow Title=Multiple
Number of Profiles=7
Profile Names=10-year,25-year,50-year,1pct_min,100-year,1pct_plu,500-year
River Rch & RM= Denton Creek Tri,Reach-1,35066
     503     672     809     483     964    1924    1371
River Rch & RM= Denton Creek Tri,Reach-1,31249
     949    1322    1633     999    1994    3979    2982
River Rch & RM= Denton Creek Tri,Reach-1,26176
    1313    1856    2316    1430    2852    5691    4342
River Rch & RM= Denton Creek Tri,Reach-1,23335
    1693    2421    3044    1892    3776    7534    5831
River Rch & RM= Denton Creek Tri,Reach-1,15895
    1992    2866    3620    2259    4507    8992    7012
River Rch & RM= Denton Creek Tri,Reach-1,7682
    2083    3004    3798    2373    4734    9445    7381
River Rch & RM= Denton Creek Tri,Reach-1,3666
    2180    3148    3985    2492    4971    9919    7766
Boundary for River Rch & Prof#=Denton Creek Tri,Reach-1,1
Up Type=0
Dn Type=3
Dn Slope=0.005
Boundary for River Rch & Prof#=Denton Creek Tri,Reach-1,2
Up Type=0
Dn Type=3
Dn Slope=0.005
Boundary for River Rch & Prof#=Denton Creek Tri,Reach-1,3
Up Type=0
Dn Type=3
Dn Slope=0.005
Boundary for River Rch & Prof#=Denton Creek Tri,Reach-1,4
Up Type=0
Dn Type=3
Dn Slope=0.005
Boundary for River Rch & Prof#=Denton Creek Tri,Reach-1,5
Up Type=0
Dn Type=3
Dn Slope=0.005
Boundary for River Rch & Prof#=Denton Creek Tri,Reach-1,6
Up Type=0
Dn Type=3
Dn Slope=0.005
Boundary for River Rch & Prof#=Denton Creek Tri,Reach-1,7
Up Type=0
Dn Type=3
Dn Slope=0.005

--- Denton Creek Tributary 17.g01 (geometry) ---

Geom Title=Existing Conditions
Program Version=4.10

River Reach=Denton Creek Tri,Reach-1
Reach XY= 30
        2327979.        7121960.      2328280.98      7119065.65
      2329234.16       7118340.2      2329130.62      7117766.04
      2329522.31      7117472.08       2329531.3      7116128.86
      2330827.96      7111449.56       2330479.2      7111194.67
      2330929.33      7110185.22      2330578.88      7108930.27
      2331229.48      7107880.16      2330681.05      7107315.84
      2331323.53      7106912.45      2331482.37      7105361.28
      2332327.35      7104354.58      2332231.24      7103715.93
      2332579.64      7103332.97      2332187.08       7102863.3
      2332332.62       7102311.5      2333327.91      7101450.36
      2333176.82      7099315.45      2332529.33      7098844.97
      2333378.69      7097244.96      2332829.61      7096320.62
      2333176.71      7095615.11      2334075.93       7095651.7
      2333829.36      7095125.16      2334577.43      7094003.96
      2334180.96      7093704.12        2334379.        7093160.

Type RM Length L Ch R = 1 ,35066   ,324,324,324
BEGIN DESCRIPTION:
Mapping XS 0ac4e1bd
END DESCRIPTION:
XS GIS Cut Line= 2
      2328736.32      7119442.53      2327934.35      7119279.35
#Sta/Elev= 30
  4482.1  775.63  4540.6  774.66  4581.4   774.8  4632.4  774.43  4683.5  774.64
  4734.5  773.91  4805.9   773.8  4877.4  772.97  4887.6  773.05    4908  772.44
  4917.1  772.67  4922.2  769.95  4938.6  770.26    4959  771.72  4972.8  771.55
  4987.6  769.83  4987.9  769.33  4991.4  769.33  4991.6  769.83  4999.8  771.39
  5030.4  771.63  5040.6  772.53    5061  775.53  5081.5  774.89  5101.9  775.19
  5112.1  776.49  5163.1  776.54  5234.5  778.14  5271.2  779.29  5300.5  779.73
#Mann= 3 ,-1 , 0
  4482.1     .05       0  4987.6     .04       0  4991.6     .05       0
Bank Sta=4987.6,4991.6
XS Rating Curve= 0 ,0
Exp/Cntr=0.3,0.1

Type RM Length L Ch R = 1 ,34742   ,348,348,348
BEGIN DESCRIPTION:
Mapping XS 10f8d9e2
END DESCRIPTION:
XS GIS Cut Line= 2
      2328886.37      7119038.08      2327982.57      7119037.03
#Sta/Elev= 30
  4413.9  771.82  4551.3  770.56  4571.3  769.63  4621.3  768.63  4651.3  768.63
  4661.3  767.79  4679.3   767.6  4679.5   767.1    4683   767.1  4683.3   767.6
  4701.3  768.54  4771.3  769.03  4821.3  768.46  4891.3  770.01  4921.3  769.71
  4961.3  770.54  4981.3  770.31  4991.3  769.11  5011.3  769.97  5051.3   769.8
  5061.3  770.53  5071.3  772.96  5091.3  774.13  5131.3  774.43  5171.3  775.44
  5191.3  776.44  5201.3  776.31  5221.3  777.52  5271.3  778.58  5317.7  780.44
#Mann= 3 ,-1 , 0
  4413.9     .05       0  4679.3    .033       0  4683.3     .05       0
Bank Sta=4679.3,4683.3
XS Rating Curve= 0 ,0
Exp/Cntr=0.3,0.1

Type RM Length L Ch R = 1 ,34394   ,353,353,353
BEGIN DESCRIPTION:
Mapping XS 62265ab8
END DESCRIPTION:
XS GIS Cut Line= 2
      2329043.47      7118929.44      2328058.56      7118895.27
#Sta/Elev= 30
  4550.3  770.64  4634.8  769.25  4674.1  769.69  4684.8  769.42  4724.9   770.1
  4794.9  767.76  4834.9  768.39    4925  767.42    4935  767.12  4968.4  765.05
    4975  765.73    4985  764.51    4993  763.97  4993.3  763.47  4996.8  763.47
    4997  763.97    5005  765.05  5045.1  764.75  5055.1  765.26  5065.1  766.79
  5075.1  769.14  5105.1  769.39  5175.1   768.7  5185.2  769.17  5205.2  769.35
  5235.2  771.59  5325.2  772.88  5355.3  773.72  5365.3  773.65  5535.8  777.86
#Mann= 3 ,-1 , 0
  4550.3     .05       0    4993    .033       0    4997     .05       0
Bank Sta=4993,4997
XS Rating Curve= 0 ,0
Exp/Cntr=0.3,0.1

Type RM Length L Ch R = 1 ,34041   ,334,334,334
BEGIN DESCRIPTION:
Mapping XS 1682fb86
END DESCRIPTION:
XS GIS Cut Line= 2
      2329034.02      7118906.22      2328437.18      7118394.78
#Sta/Elev= 30
  4706.9  770.06    4743  768.66  4757.2  768.89  4800.1  768.38  4806.6  768.77
  4814.3  768.62  4820.9  767.94  4863.7  766.98  4884.7  767.46  4935.1  765.24
  4970.2  764.42  4984.4  765.11  4998.7  763.53  5003.3  763.44  5003.6  762.94
  5007.1  762.94  5007.3  763.44    5013  764.84  5027.3  765.24  5033.8  765.18
  5041.5  764.32  5048.1  764.91  5083.2   765.4  5111.8  764.71  5161.3  765.13
  5183.1  766.12  5197.4  767.36  5218.2  767.18  5275.3  768.69  5492.9  769.91
#Mann= 3 ,-1 , 0
  4706.9     .05       0  5003.3     .04       0  5007.3     .05       0
Bank Sta=5003.3,5007.3
XS Rating Curve= 0 ,0
Exp/Cntr=0.3,0.1

Type RM Length L Ch R = 1 ,33707   ,297,297,297
BEGIN DESCRIPTION:
Mapping XS f6472d4a
END DESCRIPTION:
XS GIS Cut Line= 2
      2329305.36      7118693.36        2328647.      7118157.92
#Sta/Elev= 30
  4601.6  770.25    4673   769.1  4708.2  768.14  4736.9  768.49  4751.3  767.27
  4772.1  766.65  4906.4  763.91  4949.5  763.82  4970.7   764.4  4978.3  763.35
  4992.6  764.12    5007  764.06  5013.4  763.57  5021.4  764.09  5035.2  764.06
  5048.6  763.58  5056.6  764.25  5085.3  763.78  5089.7  763.28    5090  762.78
  5093.5  762.78  5093.7  763.28  5112.5  763.69  5126.9  764.68  5134.8  765.77
  5149.2  766.05  5190.8  765.66  5361.8  766.14  5390.5  766.69  5450.2  766.66
#Mann= 3 ,-1 , 0
  4601.6     .05       0  5089.7     .04       0  5093.7     .05       0
Bank Sta=5089.7,5093.7
XS Rating Curve= 0 ,0
Exp/Cntr=0.3,0.1

Type RM Length L Ch R = 1 ,33410   ,312,312,312
BEGIN DESCRIPTION:
Mapping XS 378c434c
END DESCRIPTION:
XS GIS Cut Line= 3
      2329325.44       7118487.5       2329105.2      7118279.97
      2328702.44      7118173.91
#Sta/Elev= 30
  4849.7  767.89  4852.5  767.23  4866.7  766.44  4937.5  764.77  4944.3  764.88
  4951.6  764.07    4978  763.33  4978.2  762.83  4981.7  762.83    4982  763.33
  5029.3  763.55  5036.6  764.53  5043.5  764.68  5071.8  764.28  5128.4  764.56
  5152.3  764.31  5158.7  764.56  5167.9  764.23  5231.1  764.87  5282.8  764.94
    5294  764.36  5329.1  764.25  5334.5  764.62  5375.9     765  5409.8   764.9
  5417.2  765.17  5479.3  765.53  5485.2  765.85    5500  765.57  5568.8  766.34
#Mann= 3 ,-1 , 0
  4849.7     .05       0    4978    .033       0    4982     .05       0
Bank Sta=4978,4982
XS Rating Curve= 0 ,0
Exp/Cntr=0.3,0.1

Type RM Length L Ch R = 1 ,33098   ,159,159,159
BEGIN DESCRIPTION:
Mapping XS a219866b
END DESCRIPTION:
XS GIS Cut Line= 5
      2329426.23      7117981.55      2329325.63      7118007.76
      2329215.34      7118057.48      2329180.21      7118114.26
      2328743.27      7118094.47
#Sta/Elev= 30
  4656.6  764.46  4674.9  764.03  4695.1  762.13  4715.7  761.51  4726.1  760.67
  4796.9  760.27  4797.1  759.77  4800.6  759.77  4800.9  760.27  4804.4  760.94
  4811.7  760.49    4822  760.86  4827.5  761.76  4850.6   761.3  4856.1  761.86
  4873.8  761.11  4902.6  761.85  4908.5  761.34    4918  762.27  4923.9  761.94
  4939.3  763.44  4969.5  763.11  4979.6  763.94  4989.6  762.19  5039.6  763.42
  5069.6  763.49  5099.7  762.76  5129.7  763.51  5159.7  763.05  5385.7  765.49
#Mann= 3 ,-1 , 0
  4656.6     .05       0  4796.9     .04       0  4800.9     .05       0
Bank Sta=4796.9,4800.9
XS Rating Curve= 0 ,0
Exp/Cntr=0.3,0.1

Type RM Length L Ch R = 1 ,32939   ,375,375,375
BEGIN DESCRIPTION:
Mapping XS 618bafd2
END DESCRIPTION:
XS GIS Cut Line= 2
      2329462.79       7117951.2      2328727.02      7117958.36
#Sta/Elev= 30
  4674.1  765.79  4727.9  763.51  4737.9  762.51  4767.9  760.53  4777.9  760.28
  4817.9  761.14  4827.9  760.69  4847.9   760.7  4857.9  759.53  4897.9  759.12
  4905.9  758.42  4906.1  757.92  4909.6  757.92  4909.9  758.42  4917.9  759.29
  4927.9  759.58  4947.9  758.87  4977.9  759.64  4997.9  759.57  5017.9  760.29
  5027.9  759.96  5047.9   760.2  5077.9  761.18  5097.9  761.06  5127.9  762.25
  5147.9  762.13  5167.9  762.62  5237.9  762.85  5247.9  763.19  5409.9  764.79
#Mann= 3 ,-1 , 0
  4674.1     .05       0  4905.9     .04       0  4909.9     .05       0
Bank Sta=4905.9,4909.9
XS Rating Curve= 0 ,0
Exp/Cntr=0.3,0.1

Type RM Length L Ch R = 1 ,32564   ,170,170,170
BEGIN DESCRIPTION:
Mapping XS b18e93ea
END DESCRIPTION:
XS GIS Cut Line= 2
      2329515.76      7117855.43      2329082.83      7117542.98
#Sta/Elev= 30
  4651.3  764.49  4673.6  764.57  4682.2  764.07  4709.2  763.87  4738.6  763.08
  4753.3  763.17  4782.8  762.46  4853.9  759.21  4860.1  758.54  4874.8  757.78
  4895.7  757.63    4946  757.93  4981.6  757.17  4990.1  756.59  4996.3  755.62
  5002.8  755.18  5003.1  754.68  5006.6  754.68  5006.8  755.18    5011  755.69
  5017.3  758.45  5025.7  758.61  5031.9  759.35  5054.3  759.62  5067.5  760.32
  5082.2  760.36  5111.6  761.42  5132.5  761.29  5140.6  760.71  5185.2  760.93
#Mann= 3 ,-1 , 0
  4651.3     .05       0  5002.8     .04       0  5006.8     .05       0
Bank Sta=5002.8,5006.8
XS Rating Curve= 0 ,0
Exp/Cntr=0.3,0.1

Type RM Length L Ch R = 1 ,32394   ,295,295,295
BEGIN DESCRIPTION:
Mapping XS 25c2c7ba
END DESCRIPTION:
XS GIS Cut Line= 2
      2329552.92      7117701.54      2329153.01      7117358.48
#Sta/Elev= 30
  4723.3  762.51  4755.1   761.6  4762.7  762.11  4797.9  761.53  4875.8  758.86
    4890  758.68  4904.3  757.99  4918.6  757.63  4947.1  757.62  4961.4  757.25
    4968  756.66  4975.6   756.8  4989.9  755.73  5004.2  752.62  5008.8  752.46
    5009  751.96  5012.5  751.96  5012.8  752.46  5018.3  754.93    5025  756.86
  5031.6  757.66  5039.3  757.87  5045.9  759.09  5060.2   759.6  5082.1     760
  5088.7  758.89  5110.6  758.82  5195.1  759.11    5216  759.46  5250.2  759.12
#Mann= 3 ,-1 , 0
  4723.3     .05       0  5008.8     .04       0  5012.8     .05       0
Bank Sta=5008.8,5012.8
XS Rating Curve= 0 ,0
Exp/Cntr=0.3,0.1

Type RM Length L Ch R = 1 ,32099   ,429,429,429
BEGIN DESCRIPTION:
Mapping XS c27dabc9
END DESCRIPTION:
XS GIS Cut Line= 2
      2329914.81      7117532.26      2329198.29      7117265.96
#Sta/Elev= 30
  4568.8  770.63    4575  770.89    4607  769.06  4761.8  762.84  4767.1  763.16
  4777.7  762.57  4822.5  761.95  4847.5  761.09  4852.8  760.34  4872.5  759.59
  4969.7  757.46  4980.4  756.16  4988.6  752.63    4994  752.89  5001.7  751.53
  5010.4  751.43  5010.6  750.93  5014.1  750.93  5014.4  751.43    5019  755.68
  5024.3  755.43  5049.3  755.99  5055.1  756.55  5074.3  756.98  5079.7  756.74
  5119.1  758.48  5165.4   758.7  5183.1  759.31  5226.1  758.53  5333.2  758.61
#Mann= 3 ,-1 , 0
  4568.8     .05       0  5010.4     .04       0  5014.4     .05       0
Bank Sta=5010.4,5014.4
XS Rating Curve= 0 ,0
Exp/Cntr=0.3,0.1

Type RM Length L Ch R = 1 ,31670   ,421,421,421
BEGIN DESCRIPTION:
Mapping XS 97259d68
END DESCRIPTION:
XS GIS Cut Line= 4
      2330069.79      7117005.91      2329542.04      7116957.57
      2329415.82      7116940.74      2329195.38      7117235.04
#Sta/Elev= 30
  4438.3  765.58  4579.7  761.82  4830.7  758.32  4870.9  758.31    4901  756.83
  4921.1  756.25  4931.1  757.05  4941.2  757.25  4967.3  753.69  4972.3  753.69
  4981.4  752.35  4987.1  750.87  4990.1  750.68  4990.4  750.18  4993.9  750.18
  4994.1  750.68  5011.7  750.74  5021.8   751.8  5031.9  753.55  5041.9   753.9
  5072.2  753.85  5107.2   754.4  5135.2  754.11    5179  754.64  5185.2  755.26
  5193.5  755.23  5207.1  755.92  5235.2  755.93  5264.4  757.04  5463.3  758.51
#Mann= 3 ,-1 , 0
  4438.3     .05       0  4990.1     .04       0  4994.1     .05       0
Bank Sta=4990.1,4994.1
XS Rating Curve= 0 ,0
Exp/Cntr=0.3,0.1

Type RM Length L Ch R = 1 ,31249   ,443,443,443
BEGIN DESCRIPTION:
Denton Creek Tributary 17 54.0
END DESCRIPTION:
XS GIS Cut Line= 3
      2330178.96        7116610.        2329529.        7116560.
      2328853.35      7116793.05
#Sta/Elev= 30
  4348.6  767.61  4368.6  766.67  4388.7  764.91  4408.7  764.09  4478.9   761.7
  4539.1  760.29  4559.2  759.19  4589.3  758.54  4629.4  758.68  4860.1  755.68
  4960.4  752.93  4970.4  752.39  4980.4  750.83  4987.6  750.72  4988.5  750.22
  4992.4  750.22  4993.3  750.72  5047.3  750.91    5064   752.1  5140.9  753.26
  5203.3  753.26  5222.6  753.64  5254.4  755.09  5286.1  754.86  5416.4  756.01
  5473.5     756    5510  756.91  5567.1  757.45    5614   757.3  5715.2  757.96
#Mann= 3 ,-1 , 0
  4348.6     .05       0  4987.6     .04       0  4993.3     .05       0
Bank Sta=4987.6,4993.3
XS Rating Curve= 0 ,0
Exp/Cntr=0.3,0.1

Type RM Length L Ch R = 1 ,30806   ,299,299,299
BEGIN DESCRIPTION:
Denton Creek Tributary 17 53.0
END DESCRIPTION:
XS GIS Cut Line= 3
       2330045.5      7116110.62      2329430.92      7116121.03
      2328613.77      7116039.15
#Sta/Elev= 30
  4489.4  756.23  4545.9  755.33  4765.9   753.2  4805.9  752.16  4855.9   750.1
    4946  748.33    4956  748.53    4976  747.07    4996  746.46  5003.1  745.45
    5004  744.95  5007.9  744.95  5008.9  745.45    5016  745.61    5036  748.57
    5046  748.91    5076  749.43  5126.1  749.15  5167.9  749.46  5296.9  751.78
    5317  752.49  5447.7  754.86  5658.7  760.24  5678.8  761.16  5749.2  763.13
  5779.3  764.51  5809.5  765.23  5859.7  767.87  5889.9  770.23  5925.3  771.04
#Mann= 3 ,-1 , 0
  4489.4     .05       0  5003.1     .04       0  5008.9     .05       0
Bank Sta=5003.1,5008.9
XS Rating Curve= 0 ,0
Exp/Cntr=0.3,0.1

Type RM Length L Ch R = 1 ,30507   ,443,443,443
BEGIN DESCRIPTION:
Denton Creek Tributary 17 52.0
END DESCRIPTION:
XS GIS Cut Line= 3
      2330239.69      7116185.52      2329551.83      7115797.42
      2328958.46      7115528.64
#Sta/Elev= 30
  4287.9  763.04  4307.6  762.08  4313.3  762.27  4329.3  760.97    4335  761.73
  4357.6  760.77  4366.8  761.03  4372.6  759.86  4388.5  759.08  4496.8  755.92
  4755.4  752.44  4814.6  751.17  4908.7  747.96  4982.1  746.85  4989.1   746.3
    4998  744.74  5009.1  744.01    5010  743.51    5014  743.51  5014.9  744.01
  5019.7  745.04  5025.4  745.16    5035  746.99  5102.5  746.98  5168.6  747.88
  5311.3  751.64  5568.8  756.26  5638.1  758.22  5666.7  758.53  5729.1  760.68
#Mann= 3 ,-1 , 0
  4287.9     .05       0  5009.1     .04       0  5014.9     .05       0
Bank Sta=5009.1,5014.9
XS Rating Curve= 0 ,0
Exp/Cntr=0.3,0.1

Type RM Length L Ch R = 1 ,30064   ,413,413,413
BEGIN DESCRIPTION:
Denton Creek Tributary 17 51.0
END DESCRIPTION:
XS GIS Cut Line= 3
      2330378.97      7116209.97        2329729.        7115410.
      2328929.01        7114960.
#Sta/Elev= 30
  3959.5     772  3987.5  771.55  3995.4     769  4001.8  768.33  4009.8   765.6
  4023.9  766.27  4051.4  765.46  4094.5  762.63  4236.7  757.43  4527.6  751.74
  4834.4  749.12  4968.7  745.16  4976.6  744.67    4983  742.79  4993.1  742.72
  4995.2   741.8  4996.2   741.3  5001.1   741.8  5013.2  742.16  5019.9  744.94
  5025.6  745.31  5063.2  745.05  5122.5  746.95  5246.8  747.32  5311.8  748.95
  5430.4  750.25  5511.3  752.13  5527.3   753.4  5775.8  759.36  5908.1  764.07
#Mann= 3 ,-1 , 0
  3959.5     .05       0  4995.2     .04       0  5001.1     .05       0
Bank Sta=4995.2,5001.1
XS Rating Curve= 0 ,0
Exp/Cntr=0.3,0.1

Type RM Length L Ch R = 1 ,29651   ,662,662,662
BEGIN DESCRIPTION:
Denton Creek Tributary 17 50.0
END DESCRIPTION:
XS GIS Cut Line= 3
      2330478.99      7115709.99        2329729.        7114910.
      2328928.98        7114910.
#Sta/Elev= 30
    4032  759.04  4053.2  758.32  4060.1  757.19  4081.6  756.35  4138.2  754.83
  4258.4   752.6  4491.9  749.54    4506  749.65  4562.7  748.54  4654.5  748.15
  4725.4  747.12  4965.7  744.75    4973  744.56  4976.9  741.25  4977.9  740.75
  4981.9  740.75  4982.9  741.25  4987.2  742.15    4994  742.66  5001.3  742.41
  5008.2  741.26  5015.5  741.49  5022.3  743.75  5036.5  743.15  5086.3  743.14
  5218.6  745.09  5378.6  748.97  5568.6  753.01  5668.6  755.58  5928.6  764.43
#Mann= 3 ,-1 , 0
    4032     .05       0  4976.9     .04       0  4982.9     .05       0
Bank Sta=4976.9,4982.9
XS Rating Curve= 0 ,0
Exp/Cntr=0.3,0.1

Type RM Length L Ch R = 1 ,28989   ,468,468,468
BEGIN DESCRIPTION:
Mapping XS c192e643
END DESCRIPTION:
XS GIS Cut Line= 2
      2330675.45      7114453.21      2329203.93      7114325.01
#Sta/Elev= 30
  4414.7  750.23  4581.8  745.03  4601.9  744.73  4611.9  745.49  4625.7  745.57
    4632  744.63  4652.1  743.19  4722.3  741.83  4732.4  741.29  4782.5  740.31
  4872.9   740.1  4983.3  740.47  4990.3  738.46  4991.3  737.96  4995.3  737.96
  4996.4  738.46  5023.5   741.3  5063.6   740.9  5073.6  741.41    5164  742.38
  5194.1  743.12  5199.9  742.87  5244.3   743.8  5485.2     746  5605.6  748.89
    5706  750.56  5716.1  751.15  5736.1  751.29    5774  752.89  5891.8  755.76
#Mann= 3 ,-1 , 0
  4414.7     .05       0  4990.3    .035       0  4996.4     .05       0
Bank Sta=4990.3,4996.4
XS Rating Curve= 0 ,0
Exp/Cntr=0.3,0.1

Type RM Length L Ch R = 1 ,28521   ,211,211,211
BEGIN DESCRIPTION:
Mapping XS b12e6d19
END DESCRIPTION:
XS GIS Cut Line= 2
      2330804.07      7113972.82      2329403.88      7113976.34
#Sta/Elev= 30
  4477.9  746.34    4693  742.54    4783  741.75    4813  742.84    4833  740.29
    4863  739.63    4953  738.74    4983  739.27    4993  736.61  4999.8  736.45
  5000.8  735.95  5005.1  735.95  5006.1  736.45    5013  739.86    5043  738.84
    5103  739.37    5183  739.24  5341.3  740.83    5353  740.58    5433     742
    5453  741.78    5473  742.31    5673  744.35    5723   746.4    5733  747.98
    5763  748.65    5813  748.38    5833  748.84    5853  748.17  5878.1  748.56
#Mann= 3 ,-1 , 0
  4477.9     .05       0  4999.8    .035       0  5006.1     .05       0
Bank Sta=4999.8,5006.1
XS Rating Curve= 0 ,0
Exp/Cntr=0.3,0.1

Type RM Length L Ch R = 1 ,28310   ,255,255,255
BEGIN DESCRIPTION:
Mapping XS c37c0ea7
END DESCRIPTION:
XS GIS Cut Line= 2
      2330666.93      7113778.54      2329338.02      7113763.59
#Sta/Elev= 30
    4682  742.61  4789.9  740.79  4829.9   740.8  4849.9  741.41  4859.9  741.12
  4869.9  739.92  4959.9  738.49    4980  736.66  4997.8  735.81  4998.8  735.31
  5004.2  735.81    5030  737.22    5050  739.72    5060  738.41    5070   738.1
    5130  737.92    5140  737.95    5160  739.85    5170   740.1    5230     740
    5270  739.44    5290  737.92    5350  740.52    5420  740.06    5600  741.58
    5720  743.11    5750  745.15    5760  744.06    5800  744.18    6011  747.94
#Mann= 3 ,-1 , 0
    4682     .05       0  4997.8     .04       0  5004.2     .05       0
Bank Sta=4997.8,5004.2
XS Rating Curve= 0 ,0
Exp/Cntr=0.3,0.1

Type RM Length L Ch R = 1 ,28055   ,456,456,456
BEGIN DESCRIPTION:
Mapping XS ccb3d3fb
END DESCRIPTION:
XS GIS Cut Line= 2
        2330668.       7113682.2      2329763.62      7113136.42
#Sta/Elev= 30
  4701.8  741.43  4775.2  740.34  4840.8  738.65  4876.1  739.04  4891.6  738.07
    4913  738.15  4922.5  736.65  4928.5  737.21  4957.6  736.48  4971.2  734.75
  5004.9  732.92  5005.9  732.42  5010.2  732.42  5011.3  732.92    5016  733.97
  5029.4   735.3  5066.3  735.89  5140.1   736.2  5161.4  735.21  5198.3  735.23
  5219.7  734.23  5235.2   734.8    5241  734.58  5249.6  735.14  5256.5  736.76
  5262.4  736.02    5272   737.5  5351.6  737.28  5431.2  738.31  5758.1  740.09
#Mann= 3 ,-1 , 0
  4701.8     .05       0  5004.9    .033       0  5011.3     .05       0
Bank Sta=5004.9,5011.3
XS Rating Curve= 0 ,0
Exp/Cntr=0.3,0.1

Type RM Length L Ch R = 1 ,27599   ,655,655,655
BEGIN DESCRIPTION:
Mapping XS 359a0462
END DESCRIPTION:
XS GIS Cut Line= 2
       2330841.6      7113229.28      2329824.89      7112874.89
#Sta/Elev= 30
  4584.9  737.23  4719.7  734.18  4781.9  733.21  4884.2  732.54  4915.9  733.06
  4926.5  733.96    4932  732.99  4937.3  732.82  4947.7  733.35    4963  733.17
  4979.5  731.37  4988.8  731.55  5008.1  729.24  5009.1  728.74  5013.5  728.74
  5014.5  729.24  5025.2  733.24  5056.3     732  5064.2  733.12  5118.4  733.28
  5175.3  734.48  5180.7  734.92  5206.4  734.64  5254.8  735.59  5361.7  735.78
  5475.5  737.36  5599.8  737.87  5614.9  738.07  5630.8  739.03  5661.6   738.6
#Mann= 3 ,-1 , 0
  4584.9     .05       0  5008.1     .04       0  5014.5     .05       0
Bank Sta=5008.1,5014.5
XS Rating Curve= 0 ,0
Exp/Cntr=0.3,0.1

Type RM Length L Ch R = 1 ,26944   ,406,406,406
BEGIN DESCRIPTION:
Denton Creek Tributary 17 44.0
END DESCRIPTION:
XS GIS Cut Line= 3
      2330990.01      7112572.76        2330529.        7112460.
      2329906.36      7112338.92
#Sta/Elev= 30
    4447  733.24  4530.4  732.41  4705.4  728.96  4839.2  728.43  4870.1  727.84
  4931.8  728.45  4938.5  724.24  4939.6  723.74  4944.3  723.74  4945.4  724.24
  4947.4  728.97  4962.3  729.29  4972.5  728.94  4982.7  727.41  4992.9  724.61
  4999.1  725.87  5004.2  725.53  5013.3  728.61  5023.5  731.26  5033.7  731.98
  5043.8  731.05  5055.8  730.72  5107.5  732.39  5159.2  731.83  5308.7  732.93
  5359.7  733.75    5380  734.97  5469.1  735.52  5525.9  734.44  5555.9  735.07
#Mann= 3 ,-1 , 0
    4447     .05       0  4938.5     .04       0  4945.4     .05       0
Bank Sta=4938.5,4945.4
XS Rating Curve= 0 ,0
Exp/Cntr=0.3,0.1

Type RM Length L Ch R = 1 ,26538   ,362,362,362
BEGIN DESCRIPTION:
Mapping XS 13ace3fe
END DESCRIPTION:
XS GIS Cut Line= 3
      2330967.05      7112367.04      2330710.81      7112107.91
      2330216.37       7112050.4
#Sta/Elev= 30
  4494.3  730.75  4533.2   730.7  4632.2  727.55  4717.1  725.97  4752.5  725.57
  4801.9  725.64  4823.2  725.05  4830.2  725.34  4910.9  725.09  4941.1  725.65
  4973.4   724.7    4988   721.6  4989.1   721.1  4993.8   721.1  4994.9   721.6
  5011.6   724.6  5031.7  724.61  5041.8  725.48  5051.8   727.4    5062  727.98
    5072   729.1    5082  729.51  5092.1  729.03  5102.2  730.27  5192.8   730.6
  5212.9  731.14  5317.6   731.6  5323.6  731.95  5343.8  731.91  5356.5  732.28
#Mann= 3 ,-1 , 0
  4494.3     .05       0    4988     .04       0  4994.9     .05       0
Bank Sta=4988,4994.9
XS Rating Curve= 0 ,0
Exp/Cntr=0.3,0.1

Type RM Length L Ch R = 1 ,26176   ,558,558,558
BEGIN DESCRIPTION:
Denton Creek Tributary 17 43.0
END DESCRIPTION:
XS GIS Cut Line= 3
      2331401.88      7111690.86      2330721.88      7111814.79
      2330199.93      7111871.25
#Sta/Elev= 30
  4316.5  743.66  4441.4  738.72  4532.9  734.12  4644.7   731.6  4654.9  730.53
  4672.2  729.59  4788.9  726.57  4837.1  724.55  4888.7  723.29  4900.6  722.62
  4929.3  723.29  4980.1  722.84  4990.3  722.53  5000.5  721.45  5006.6  721.46
  5007.7  720.26  5009.1  719.76  5016.2  719.76  5017.6  720.26  5020.7   722.6
  5030.7     723  5040.8  720.28  5050.8   722.5  5104.4  723.21  5151.4   727.3
  5241.9  729.86    5252  729.34  5262.1  730.44  5287.9  729.75  5532.7  731.38
#Mann= 3 ,-1 , 0
  4316.5     .05       0  5007.7    .033       0  5017.6     .05       0
Bank Sta=5007.7,5017.6
XS Rating Curve= 0 ,0
Exp/Cntr=0.3,0.1

Type RM Length L Ch R = 1 ,25618   ,903,903,903
BEGIN DESCRIPTION:
Denton Creek Tributary 17 42.0
END DESCRIPTION:
XS GIS Cut Line= 3
        2331179.        7111360.      2330835.13      7111327.78
      2330062.22      7111592.01
#Sta/Elev= 30
  4648.1  744.96  4668.2  744.15  4688.3  737.94  4828.9  730.48  4889.1  728.35
  4899.2  726.98  4979.5  724.38    4989  721.95  4993.5  721.95  5010.8  716.95
  5012.2  716.45  5020.8  716.95  5021.1  718.05  5041.8  720.34  5078.4  720.07
  5084.5  721.19  5126.8  720.43  5147.9  721.62  5172.3  721.54  5203.7  719.16
    5243  723.63  5328.9  726.94  5412.1  727.31  5433.2  728.57  5480.2  728.06
  5568.8  728.58  5600.1  729.11  5605.4  730.27  5623.5  730.74  5810.3  730.92
#Mann= 3 ,-1 , 0
  4648.1     .05       0  5010.8     .04       0  5020.8     .05       0
Bank Sta=5010.8,5020.8
XS Rating Curve= 0 ,0
Exp/Cntr=0.3,0.1

Type RM Length L Ch R = 1 ,24715   ,446,446,446
BEGIN DESCRIPTION:
Denton Creek Tributary 17 41.0
END DESCRIPTION:
XS GIS Cut Line= 3
      2331005.57      7110938.39      2330630.61      7110868.36
      2329983.52      7110951.06
#Sta/Elev= 30
  4615.9  727.06  4714.1  724.68  4775.2  722.36  4815.9  721.66    4826  722.12
  4836.2  720.44  4904.5  718.72  4962.3  718.69  4978.6  719.33  4988.8  715.68
  4990.6  714.18    4992  713.68  4999.3  713.68  5000.7  714.18  5009.1  715.08
  5019.1  714.65  5029.2  716.24  5069.5  716.81  5079.6   717.6  5099.8   716.9
  5126.8  720.06  5150.2  721.86  5180.4  722.89  5190.5  722.49  5206.6  723.82
  5230.8  723.78  5240.9   724.6  5261.1  724.22  5351.8  724.81  5649.7  727.92
#Mann= 3 ,-1 , 0
  4615.9     .05       0  4990.6    .033       0  5000.7     .05       0
Bank Sta=4990.6,5000.7
XS Rating Curve= 0 ,0
Exp/Cntr=0.3,0.1

Type RM Length L Ch R = 1 ,24269   ,459,459,459
BEGIN DESCRIPTION:
Denton Creek Tributary 17 40.0
END DESCRIPTION:
XS GIS Cut Line= 3
      2331078.98      7110959.98      2330628.18      7110567.05
      2330373.64      7110446.62
#Sta/Elev= 30
  4400.2  729.27  4421.5  729.01    4450  727.58  4626.6  724.45  4691.2  722.49
    4712   722.3  4718.7  722.72  4726.3  721.28  4754.8  719.61  4789.9  718.99
  4832.6  717.23  4861.1  717.74  4910.5   716.9  4917.5  715.98  4959.8   714.4
  4962.3  713.83  4963.8  713.33  4971.1  713.33  4972.5  713.83  5071.2  714.23
  5076.7  715.29  5093.9   716.8  5099.5  718.49  5174.3  720.84  5207.5  721.17
  5213.2  722.05  5229.6  722.67  5241.5   722.6  5251.7  721.56  5279.8  722.23
#Mann= 3 ,-1 , 0
  4400.2     .05       0  4962.3    .033       0  4972.5     .05       0
Bank Sta=4962.3,4972.5
XS Rating Curve= 0 ,0
Exp/Cntr=0.3,0.1

Type RM Length L Ch R = 1 ,23810   ,475,475,475
BEGIN DESCRIPTION:
Denton Creek Tributary 17 39.0
END DESCRIPTION:
XS GIS Cut Line= 3
      2331278.97      7110459.98      2330862.69      7110236.68
      2330523.22      7110202.31
#Sta/Elev= 30
  4518.1  728.13    4592  725.21  4635.8   724.6  4745.4  719.77  4835.8  718.93
  4881.2  717.96  4893.2   718.3  4909.5  717.33  4947.7   712.4  4953.3     712
  4975.3  712.65  4983.3  712.12  4989.7  710.75  4994.9  710.75  4998.1  710.01
  4999.5  709.51  5006.9  709.51  5008.3  710.01  5024.4  712.35  5034.4  713.24
  5044.5  715.19  5084.7  714.34  5114.8  716.15  5134.9  716.23  5195.2     718
  5225.4  718.21  5235.4  719.24  5245.5  719.51  5255.5  718.83  5331.7  719.28
#Mann= 3 ,-1 , 0
  4518.1     .05       0  4998.1     .04       0  5008.3     .05       0
Bank Sta=4998.1,5008.3
XS Rating Curve= 0 ,0
Exp/Cntr=0.3,0.1

Type RM Length L Ch R = 1 ,23335   ,487,487,487
BEGIN DESCRIPTION:
Denton Creek Tributary 17 38.0
END DESCRIPTION:
XS GIS Cut Line= 3
      2331278.97        7109860.        2330929.        7109810.
      2330144.91      7109599.78
#Sta/Elev= 30
  4646.5  726.17  4888.9   718.9  4909.1  717.53  4949.5  712.17  4979.8  711.37
  4989.9  710.13  5031.1   710.2  5057.5  713.58  5196.7  714.52  5207.1  714.49
  5212.3  713.15  5217.5  713.49  5227.8  712.49  5238.1  710.16    5264  709.93
  5265.5  709.43  5274.4  709.93  5279.6  709.98  5287.2  711.61  5292.4  710.59
  5300.3  712.86  5327.2  715.42  5372.7  715.37  5487.3  718.05  5516.9  718.05
    5528  720.01  5548.7  719.35  5556.9   720.6  5642.1  720.37  5811.8  722.02
#Mann= 3 ,-1 , 0
  4646.5     .05       0    5264    .033       0  5274.4     .05       0
Bank Sta=5264,5274.4
XS Rating Curve= 0 ,0
Exp/Cntr=0.3,0.1

Type RM Length L Ch R = 1 ,22848   ,396,396,396
BEGIN DESCRIPTION:
Denton Creek Tributary 17 37.0
END DESCRIPTION:
XS GIS Cut Line= 3
      2331628.99        7109710.        2330829.        7109360.
      2329629.03      7109659.99
#Sta/Elev= 30
  4126.8   740.1  4164.6  736.96  4234.8  733.54  4315.9  731.14  4409.4  726.77
  4589.5  721.52  4717.4  716.69  4735.3   717.3  4764.2  715.99  4847.2  714.29
  4967.6  712.94  4978.2  713.22  5002.6  711.82  5010.3  710.38    5018  710.09
    5067  709.88  5068.4  709.38  5075.9  709.38  5077.4  709.88  5105.7  710.03
  5146.9  711.99  5224.2  713.31  5319.5  716.89  5394.3  718.07  5435.5  719.93
  5443.2  719.38  5494.8  719.58  5930.3  724.46  6102.9  727.11  6236.9   730.5
#Mann= 3 ,-1 , 0
  4126.8     .05       0    5067    .033       0  5077.4     .05       0
Bank Sta=5067,5077.4
XS Rating Curve= 0 ,0
Exp/Cntr=0.3,0.1

Type RM Length L Ch R = 1 ,22452   ,147,147,147
BEGIN DESCRIPTION:
Mapping XS 276bbecb
END DESCRIPTION:
XS GIS Cut Line= 3
      2331266.61       7109049.4      2330648.96      7109066.67
      2330165.09      7109102.78
#Sta/Elev= 30
  4369.5  716.73  4497.2  714.72  4571.1  714.44  4577.2  714.01  4587.2  714.26
  4657.2  713.16  4677.2  713.62  4697.2  712.93  4727.2  713.64  4777.3  712.72
  4807.3  713.12  4817.3  712.74  4837.3  710.07  4977.3  710.23  5001.7  709.64
  5003.3  709.14  5011.6  709.14  5013.2  709.64  5017.4  710.95    5101  711.22
  5137.8  712.48  5197.9  713.69    5218  715.64    5228  715.98  5238.4  715.62
  5248.1  716.66  5298.2   716.9  5370.7  718.44  5418.5  718.23  5472.6  718.69
#Mann= 3 ,-1 , 0
  4369.5     .05       0  5001.7    .033       0  5013.2     .05       0
Bank Sta=5001.7,5013.2
XS Rating Curve= 0 ,0
Exp/Cntr=0.3,0.1

Type RM Length L Ch R = 1 ,22305   ,537,537,537
BEGIN DESCRIPTION:
Mapping XS f6db2351
END DESCRIPTION:
XS GIS Cut Line= 2
      2331180.54      7108930.68      2330166.84      7108950.42
#Sta/Elev= 30
  4397.5   714.2  4439.1   713.7  4469.1  712.55  4529.1  712.19  4709.1  711.46
  4749.1  712.15  4789.1  710.37  4829.1  706.73  4873.4     705  4874.9   704.5
  4883.3   704.5  4884.9     705  4889.1  706.68  4899.1  708.01  4909.1   708.7
  4939.1  709.08  4949.1  710.95  4959.2   710.4  4979.2  706.25  4989.2   705.1
  5009.2  705.66  5019.2  708.02  5049.2  711.09  5128.5  714.39  5139.2  714.09
  5169.2  715.94  5179.2  715.51  5189.2   716.4  5219.2  716.16  5411.4  717.75
#Mann= 3 ,-1 , 0
  4397.5     .05       0  4873.4    .033       0  4884.9     .05       0
Bank Sta=4873.4,4884.9
XS Rating Curve= 0 ,0
Exp/Cntr=0.3,0.1

Type RM Length L Ch R = 1 ,21768   ,142,142,142
BEGIN DESCRIPTION:
Mapping XS ec1e3616
END DESCRIPTION:
XS GIS Cut Line= 2
      2331509.58      7108550.68       2330481.1      7108524.97
#Sta/Elev= 30
    4345  715.33  4705.7  709.47  4725.7   709.8  4735.7  709.06  4755.7  709.39
  4865.7  707.62  4885.8  708.02  4915.8  707.39  4925.8  707.91  4945.8  707.15
  4955.8  705.53  4965.8     705  4976.6  705.59  5015.8  704.62  5025.8  703.92
    5030  700.78  5031.6  700.28    5040  700.28  5041.6  700.78  5055.8  704.28
  5075.8  706.41  5155.8  710.69  5165.8  712.14  5175.8  712.66  5255.9  714.79
  5275.9  714.31  5305.9  715.29  5325.9  714.73  5355.9  715.95  5373.8  715.86
#Mann= 3 ,-1 , 0
    4345     .05       0    5030     .04       0  5041.6     .05       0
Bank Sta=5030,5041.6
XS Rating Curve= 0 ,0
Exp/Cntr=0.3,0.1

Type RM Length L Ch R = 1 ,21626   ,331,331,331
BEGIN DESCRIPTION:
Mapping XS 6586c7e2
END DESCRIPTION:
XS GIS Cut Line= 2
      2331431.76      7108424.98      2330544.49      7108417.33
#Sta/Elev= 30
  4497.7  712.35  4570.5  711.12  4620.5  709.42  4660.5  709.12  4670.5  710.37
  4680.5  709.06  4700.5  708.42  4770.5  707.71  4790.5   706.9  4840.5  707.96
  4850.5  706.74  4920.5  705.71  4930.5  705.97  4950.5  707.74  4960.5  707.21
  4970.5  704.87  4990.5  704.72  5000.5  700.66  5024.7  700.62  5026.3  700.12
  5034.7  700.12  5036.3  700.62  5040.5  703.39  5070.5  704.56  5120.5  708.94
  5130.5  709.15  5170.5  712.46  5290.5  714.61  5340.5  716.74    5385  716.54
#Mann= 3 ,-1 , 0
  4497.7     .05       0  5024.7     .04       0  5036.3     .05       0
Bank Sta=5024.7,5036.3
XS Rating Curve= 0 ,0
Exp/Cntr=0.3,0.1

Type RM Length L Ch R = 1 ,21295   ,512,512,512
BEGIN DESCRIPTION:
Mapping XS d9db8377
END DESCRIPTION:
XS GIS Cut Line= 3
      2331512.45        7108294.      2331037.02      7108126.15
      2330448.22      7108173.67
#Sta/Elev= 30
  4488.5  712.11  4704.3  707.85  4746.7  707.62  4753.9  706.48  4799.7   705.5
  4815.8   706.2  4831.5  705.17  4841.4  705.55  4872.3  704.12  4939.5  704.82
  4948.2  705.89  4965.1  705.68  4992.7  703.53  4994.9  700.07  4996.5  699.57
  5004.9  699.57  5006.5  700.07  5010.8  702.82  5020.8   704.8  5030.8  704.06
    5091  703.47  5099.4  700.29  5131.2  705.04  5151.2  710.07  5341.8  712.27
  5442.2  714.86  5492.3  714.36  5522.4  715.97  5552.5  715.28  5583.4  715.96
#Mann= 3 ,-1 , 0
  4488.5     .05       0  4994.9    .033       0  5006.5     .05       0
Bank Sta=4994.9,5006.5
XS Rating Curve= 0 ,0
Exp/Cntr=0.3,0.1

Type RM Length L Ch R = 1 ,20783   ,665,665,665
BEGIN DESCRIPTION:
Mapping XS 12f29107
END DESCRIPTION:
XS GIS Cut Line= 3
       2331599.4      7107791.01      2331084.98       7107738.1
      2330372.84      7107755.94
#Sta/Elev= 30
  4508.4  708.36  4689.8  706.64  4780.2  706.51  4790.3  707.17  4830.5  706.27
  4890.8  706.49  4900.9  706.26    4921  699.41  4941.1  698.58  4951.1  700.32
  4956.3  698.57    4958  698.07    4968  698.57  4991.3  700.03  5011.4  700.11
  5025.5  699.14  5041.5  701.91  5141.6   701.1  5191.6  702.61  5261.6  702.04
  5311.6  704.25  5331.6  703.45  5411.6  707.36  5491.7  710.08  5541.7  713.33
  5671.7  718.01  5691.7  719.85  5703.5  720.01  5711.7  721.49  5737.9  722.08
#Mann= 3 ,-1 , 0
  4508.4     .05       0  4956.3    .033       0    4968     .05       0
Bank Sta=4956.3,4968
XS Rating Curve= 0 ,0
Exp/Cntr=0.3,0.1

Type RM Length L Ch R = 1 ,20118   ,435,435,435
BEGIN DESCRIPTION:
Mapping XS 09b8ca5e
END DESCRIPTION:
XS GIS Cut Line= 2
      2331749.95      7107685.32      2330462.75       7107320.5
#Sta/Elev= 30
  3886.6  709.04  4043.5  706.55  4221.6  704.84  4313.7   705.6  4448.9  704.85
  4708.7  701.36  4781.5  701.62  4791.9  702.23    4806   701.1  4845.1  700.33
  4895.8  700.59    4927  699.55    4986  699.41  4991.2  698.17  5004.3  697.86
  5005.9  697.36  5014.4  697.36    5016  697.86  5030.9  698.51  5041.3   701.3
  5059.1  709.54  5072.5  712.39  5082.9  713.52    5093  714.34  5098.2  713.88
  5124.5  715.75  5137.3  715.34    5166  716.54  5171.3  717.23  5224.5  719.61
#Mann= 3 ,-1 , 0
  3886.6     .05       0  5004.3     .04       0    5016     .05       0
Bank Sta=5004.3,5016
XS Rating Curve= 0 ,0
Exp/Cntr=0.3,0.1

Type RM Length L Ch R = 1 ,19683   ,580,580,580
BEGIN DESCRIPTION:
Mapping XS 07320d84
END DESCRIPTION:
XS GIS Cut Line= 3
      2331696.91      7107546.21      2331182.38      7107323.95
      2330733.33      7106847.76
#Sta/Elev= 30
  4108.5  707.06    4334  704.36  4391.9  702.84  4438.9  704.04  4574.6  704.49
  4730.6  700.65  4773.1  700.45  4780.4  699.02  4787.2  699.25  4801.4   697.5
  4843.9  697.58  4886.4  702.43  4893.6  700.87  4900.5  701.92  4907.8  697.79
  4929.9  697.48  4931.5  696.98  4941.6  697.48    4943  698.17  4985.5  697.88
  4992.3  698.94  4999.6  703.08  5006.5  704.84  5013.8  705.51  5056.3  705.79
  5070.4  703.87  5077.3  703.74  5127.1  706.02  5183.3  707.48  5323.5  709.12
#Mann= 3 ,-1 , 0
  4108.5     .05       0  4929.9     .04       0  4941.6     .05       0
Bank Sta=4929.9,4941.6
XS Rating Curve= 0 ,0
Exp/Cntr=0.3,0.1

Type RM Length L Ch R = 1 ,19103   ,542,542,542
BEGIN DESCRIPTION:
Mapping XS 43e0791d
END DESCRIPTION:
XS GIS Cut Line= 2
      2331737.18      7106880.02      2330854.61      7106683.91
#Sta/Elev= 30
  4581.7  703.33  4692.2  700.99  4702.8  700.31  4866.7   698.6  4887.2  697.82
  4907.6  697.87  4925.3  699.08  4938.4  699.18  4958.9  695.75  4979.4  694.54
  4999.8  694.58  5010.1  692.26  5016.7  691.58  5018.4  691.08  5026.9  691.08
  5028.5  691.58  5030.6  694.63  5040.8  693.98  5071.5   696.6    5133  697.43
  5250.5  701.73  5276.4  703.28  5299.2  703.51  5317.4  704.63  5386.3   705.8
  5399.4  705.53  5419.8  706.64  5434.9  706.26  5471.1  707.21  5485.8  706.87
#Mann= 3 ,-1 , 0
  4581.7     .05       0  5016.7    .033       0  5028.5     .05       0
Bank Sta=5016.7,5028.5
XS Rating Curve= 0 ,0
Exp/Cntr=0.3,0.1

Type RM Length L Ch R = 1 ,18561   ,179,179,179
BEGIN DESCRIPTION:
Mapping XS b5e0e872
END DESCRIPTION:
XS GIS Cut Line= 2
       2331984.7      7106242.15      2330892.82       7106316.3
#Sta/Elev= 30
    4443  703.98  4448.7  703.17  4518.9  703.17  4628.4  700.92  4639.2  701.39
  4739.4  699.26  4749.4  699.64  4782.4  697.98  4809.3   698.1  4879.7  696.53
  4889.7  695.53  4899.8  693.43  4908.7  692.89  4939.8  691.64  4979.9  691.71
    4994  688.53  4995.7  688.03  5005.9  688.53    5010  691.35    5020  692.57
  5030.1  692.21  5040.1  694.15  5050.1  695.04  5070.1  694.93  5075.3  695.82
  5140.3   696.8  5170.4  698.07  5360.8  700.12    5461  704.44  5537.4   705.1
#Mann= 5 ,-1 , 0
    4443     .05       0  4809.3     .12       0  4908.7     .05       0
    4994     .04       0  5005.9     .05       0
Bank Sta=4994,5005.9
XS Rating Curve= 0 ,0
Exp/Cntr=0.3,0.1

Type RM Length L Ch R = 1 ,18382   ,285,285,285
BEGIN DESCRIPTION:
Mapping XS a9a5d149
END DESCRIPTION:
XS GIS Cut Line= 2
      2331909.62      7106115.77      2330878.63      7106173.39
#Sta/Elev= 30
  4618.7   701.9  4689.4  700.71  4757.5  698.58  4806.7  697.61  4839.7  696.95
  4859.7  697.64  4869.7  696.57  4906.1  695.02  4939.8  692.76  4979.9  692.26
  5005.4  689.67    5014  688.78  5015.6  688.28  5025.9  688.78    5040  693.12
    5050  694.43    5070  695.21  5100.1  694.53  5110.1  693.61  5120.1  694.36
  5170.2   694.4  5300.4  697.17  5318.6  696.74  5323.6  697.78  5330.4  697.25
  5420.6  699.41  5440.6  699.02  5510.7  701.46  5570.8  702.19  5651.3  705.15
#Mann= 7 ,-1 , 0
  4618.7     .05       0  4757.5     .12       0  4806.7     .05       0
  4906.1     .12       0  5005.4     .05       0    5014     .07       0
  5025.9     .05       0
Bank Sta=5014,5025.9
XS Rating Curve= 0 ,0
Exp/Cntr=0.3,0.1

Type RM Length L Ch R = 1 ,18097   ,472,472,472
BEGIN DESCRIPTION:
Mapping XS 28fbedd5
END DESCRIPTION:
XS GIS Cut Line= 2
      2331988.58      7105895.89      2330912.84      7105823.21
#Sta/Elev= 30
  4589.5  701.44  4839.7  694.88  4859.7  695.29  4897.1  694.77  4909.8  693.88
  4923.8  694.35    4933  694.38  4939.9  693.77  4949.9  690.51    4954  687.48
  4955.6  686.98  4965.9  687.48    4980  687.77    4990  689.03  5046.5  692.59
  5051.5  692.04  5070.2   692.7  5080.2  693.98  5100.2  692.58  5130.3  692.61
  5310.7  694.97    5451  698.17  5471.1  699.27  5494.5   699.4  5551.3   701.7
  5571.3  701.85  5581.3  702.69  5638.8  703.93  5643.8  704.64  5667.7  705.39
#Mann= 5 ,-1 , 0
  4589.5     .05       0  4923.8     .12       0    4933     .05       0
    4954    .033       0  4965.9     .05       0
Bank Sta=4954,4965.9
XS Rating Curve= 0 ,0
Exp/Cntr=0.3,0.1

Type RM Length L Ch R = 1 ,17625   ,369,369,369
BEGIN DESCRIPTION:
Mapping XS 50e5a643
END DESCRIPTION:
XS GIS Cut Line= 3
      2331915.54      7105596.39      2331103.45       7105284.2
      2331049.06      7105261.93
#Sta/Elev= 30
  4531.6   697.2  4752.9   692.2  4827.9  691.07    4860  691.35  4881.4  690.72
  4897.6  689.45  4982.3  689.46  4999.3  687.99  5020.7  686.99  5025.5  685.43
  5027.1  684.93  5035.7  684.93  5037.4  685.43  5042.3  689.53  5061.6  692.63
  5066.9  691.75  5074.3  693.63  5116.2  693.93  5206.3  696.19  5224.3  697.11
  5230.9  698.44  5236.3  697.83  5245.7  698.49  5260.9  698.58  5267.1  698.01
  5285.6  698.95    5385  701.22  5400.2  702.12  5453.7  703.29  5460.4  703.83
#Mann= 3 ,-1 , 0
  4531.6     .05       0  5025.5    .033       0  5037.4     .05       0
Bank Sta=5025.5,5037.4
XS Rating Curve= 0 ,0
Exp/Cntr=0.3,0.1

Type RM Length L Ch R = 1 ,17256   ,438,438,438
BEGIN DESCRIPTION:
Mapping XS c22e9798
END DESCRIPTION:
XS GIS Cut Line= 2
      2331986.76      7105415.38      2331326.63      7104866.83
#Sta/Elev= 30
  4604.6  696.25  4614.5  696.04    4621  697.15    4664  696.63  4670.5  695.61
  4684.8  695.36  4742.1   695.4  4748.6  696.01  4855.4  692.12  4912.7  692.16
  4954.3  687.28  4962.2  687.16  4968.7  684.54    4977  684.51  4978.7  684.01
    4989  684.51  4990.8   686.2  4997.3  686.96  5032.5   687.7  5068.9  690.29
  5110.6  689.36  5196.5  690.61  5231.7   690.3  5338.4  693.16  5367.1  694.57
  5373.6  696.39  5381.4  696.58  5387.9  699.33  5394.8  699.79  5462.9  700.57
#Mann= 3 ,-1 , 0
  4604.6     .05       0    4977    .033       0    4989     .05       0
Bank Sta=4977,4989
XS Rating Curve= 0 ,0
Exp/Cntr=0.3,0.1

Type RM Length L Ch R = 1 ,16818   ,405,405,405
BEGIN DESCRIPTION:
Mapping XS 05025829
END DESCRIPTION:
XS GIS Cut Line= 2
      2332189.23      7105218.52       2331579.2      7104428.16
#Sta/Elev= 30
  4451.9  694.83  4472.9  694.56  4493.7  694.84    4529  694.25    4558  693.35
  4628.7   692.1    4693  690.04  4778.5  688.16  4850.6  687.43  4914.9  687.87
  4929.4  688.55  4942.7  686.89  4950.2   686.6  4956.5  685.17  4964.7  685.64
  4979.2  685.33  4985.5  683.39    5000  684.32  5000.4  683.04  5002.1  682.54
  5010.7  682.54  5012.4  683.04  5020.9  685.31  5043.5  684.69  5085.2  687.09
  5143.2  688.11  5234.6  691.91  5271.1  692.96  5298.9  693.59  5450.3  695.44
#Mann= 3 ,-1 , 0
  4451.9     .05       0  5000.4     .04       0  5012.4     .05       0
Bank Sta=5000.4,5012.4
XS Rating Curve= 0 ,0
Exp/Cntr=0.3,0.1

Type RM Length L Ch R = 1 ,16413   ,518,518,518
BEGIN DESCRIPTION:
Mapping XS ba63bced
END DESCRIPTION:
XS GIS Cut Line= 3
      2332318.43      7105064.14      2332182.52      7104525.86
      2331742.48      7104283.58
#Sta/Elev= 30
  4319.9  694.15  4561.4  689.96    4580  689.45  4585.1  688.89  4674.8  687.17
  4736.7  686.32  4850.2  686.21  4867.3  684.98  4890.5  684.45  4896.9  684.69
  4902.6  684.03  4970.4  683.84  4978.3  683.48    4984  682.25  4993.2   682.4
  4994.1  682.07  4995.8  681.57  5004.5  681.57  5006.1  682.07  5021.9  682.18
  5027.6  684.77    5038  686.09  5065.5  686.42  5087.2  687.62  5168.7  687.76
  5184.7  688.37  5293.6  690.05  5331.5  691.28  5375.1  691.93  5377.4  692.34
#Mann= 3 ,-1 , 0
  4319.9     .05       0  4994.1     .04       0  5006.1     .05       0
Bank Sta=4994.1,5006.1
XS Rating Curve= 0 ,0
Exp/Cntr=0.3,0.1

Type RM Length L Ch R = 1 ,15895   ,361,361,361
BEGIN DESCRIPTION:
Mapping XS 4a11c76b
END DESCRIPTION:
XS GIS Cut Line= 2
      2332794.98      7104143.21      2331746.04      7104161.64
#Sta/Elev= 30
    4484  692.56    4520  691.25    4540  690.96    4560  690.05    4600  689.15
    4680  686.86    4730   685.8    4800  685.56    4860  685.05    4900  685.24
  4960.1  685.19  4970.1  683.31  4973.9  680.57  4975.6  680.07  4984.5  680.07
  4986.3  680.57  5000.1  680.81  5070.1  683.18  5080.1  683.36  5120.1  683.31
  5190.1  684.13  5200.1  684.34  5210.1   684.9  5230.1   685.3  5260.1  685.29
  5330.1  686.37  5350.1  686.82  5390.1  688.37  5480.1  691.37  5533.1  692.59
#Mann= 3 ,-1 , 0
    4484     .05       0  4973.9     .04       0  4986.3     .05       0
Bank Sta=4973.9,4986.3
XS Rating Curve= 0 ,0
Exp/Cntr=0.3,0.1

Type RM Length L Ch R = 1 ,15534   ,632,632,632
BEGIN DESCRIPTION:
Mapping XS 4603deea
END DESCRIPTION:
XS GIS Cut Line= 3
      2332910.99      7103863.15      2332161.88      7103802.63
       2331743.7      7103964.05
#Sta/Elev= 30
  4315.7  693.58  4347.8   693.2  4357.8  692.01  4377.9  690.96  4428.1   689.9
  4537.3  686.64  4542.3  686.89  4669.6  682.82  4799.3  682.07  4849.4  682.45
  4969.8  681.05  4989.9  679.91  5013.7  676.72  5015.4  676.22  5024.5  676.22
  5026.3  676.72    5030  679.09  5036.5  681.49  5041.5  681.63  5060.1   685.2
  5066.2  685.78  5104.7  685.84  5183.9  688.26  5213.9  688.37  5238.5  687.32
  5263.1  686.86  5316.9   686.9  5391.9   687.8  5456.2  689.37  5515.5     690
#Mann= 3 ,-1 , 0
  4315.7     .05       0  5013.7    .033       0  5026.3     .05       0
Bank Sta=5013.7,5026.3
XS Rating Curve= 0 ,0
Exp/Cntr=0.3,0.1

Type RM Length L Ch R = 1 ,14902   ,522,522,522
BEGIN DESCRIPTION:
Mapping XS 89bcc9ae
END DESCRIPTION:
XS GIS Cut Line= 3
      2332912.07      7103443.26      2332578.38      7103331.27
      2331813.02      7103154.01
#Sta/Elev= 30
  4649.3  688.98  4874.1  683.27  4937.3  682.84    4969   683.3  4987.2  680.55
  4992.5  680.32  4998.3  677.11  5003.5  677.11  5004.6  675.31  5006.4  674.81
  5015.5  674.81  5017.2  675.31  5027.7  676.48  5032.8   675.8  5041.7  678.09
    5052  677.99  5070.4  678.77  5134.1  679.48  5208.7  678.93  5341.9  680.63
  5370.2  683.18  5379.5  685.41  5421.5  685.08  5483.1     686  5517.8  686.03
  5554.9  687.41  5626.8  688.41  5645.9  689.26  5741.5  690.15  5786.9  691.07
#Mann= 3 ,-1 , 0
  4649.3     .05       0  5004.6     .04       0  5017.2     .05       0
Bank Sta=5004.6,5017.2
XS Rating Curve= 0 ,0
Exp/Cntr=0.3,0.1

Type RM Length L Ch R = 1 ,14380   ,298,298,298
BEGIN DESCRIPTION:
Mapping XS c7b6f1ce
END DESCRIPTION:
XS GIS Cut Line= 2
      2332905.21      7102892.58       2332002.8      7103004.27
#Sta/Elev= 30
  4318.4  683.47  4338.9  683.51  4395.2  682.43  4495.9   681.5  4596.7  681.12
  4647.1  680.29  4717.6  679.91    4825   677.4  4848.6  677.73  4878.9  678.81
  4888.9  678.08    4911  678.05  4979.6  676.01    4987  673.74  4993.5  672.49
  4995.2  671.99  5004.3  671.99  5006.1  672.49  5009.8  672.76    5030  678.55
  5040.1  679.68  5050.2  679.52  5060.2  679.92    5068  681.52  5073.1  684.25
  5080.4  684.54  5110.6  684.08  5140.8   684.8  5171.1  684.93  5227.7  686.73
#Mann= 3 ,-1 , 0
  4318.4     .05       0  4993.5    .033       0  5006.1     .05       0
Bank Sta=4993.5,5006.1
XS Rating Curve= 0 ,0
Exp/Cntr=0.3,0.1

Type RM Length L Ch R = 1 ,14082   ,273,273,273
BEGIN DESCRIPTION:
Mapping XS 76b1435f
END DESCRIPTION:
XS GIS Cut Line= 2
      2332905.24      7102700.38      2331963.77      7102707.89
#Sta/Elev= 30
  4323.8  682.57    4390  681.26    4430  681.04    4450  680.37    4580  678.23
    4640  678.26  4670.1  677.64  4710.1  677.46  4730.1  677.65  4810.1  676.33
  4860.1  676.36  4880.1  676.75  4898.9  677.83  4903.9  677.73  4920.1  676.31
  4930.1  676.92  4950.1  676.32  4960.1  674.82  4993.8   672.4  4995.5   671.9
  5004.6   671.9  5006.4   672.4  5010.1  674.59  5020.1  674.86  5030.1  675.96
  5050.1  680.01  5070.1  681.49  5190.1  685.67  5240.1  686.75  5265.3  687.86
#Mann= 3 ,-1 , 0
  4323.8     .05       0  4993.8     .04       0  5006.4     .05       0
Bank Sta=4993.8,5006.4
XS Rating Curve= 0 ,0
Exp/Cntr=0.3,0.1

Type RM Length L Ch R = 1 ,13809   ,144,144,144
BEGIN DESCRIPTION:
Mapping XS bed8978a
END DESCRIPTION:
XS GIS Cut Line= 3
      2332929.95      7102446.12      2332515.01      7102431.04
       2332029.5      7102474.89
#Sta/Elev= 30
  4358.3     681  4449.3   679.8  4469.3  679.89  4489.3  679.48  4499.3  678.78
  4519.4   678.2  4549.4  678.73  4659.4  677.28  4869.9  675.33    4880  675.29
    4900  675.84  4920.1  675.81  4926.9  675.18    4932  675.45  4940.2  674.42
  4950.2  674.93  4980.4  674.24  4990.4   674.7  4994.1  672.48  4995.9  671.98
    5005  671.98  5006.8  672.48  5020.5  672.58  5030.6  674.24  5037.8  676.36
  5042.8  675.44  5060.7  681.12  5070.7  682.41  5110.9  683.89    5261  687.16
#Mann= 3 ,-1 , 0
  4358.3     .05       0  4994.1    .033       0  5006.8     .05       0
Bank Sta=4994.1,5006.8
XS Rating Curve= 0 ,0
Exp/Cntr=0.3,0.1
