--- MDW T 021.prj (project) ---

Proj Title=MDW T 021 Base Level Engineering
Current Plan=p01
Default Exp/Contr=0.3,0.1
English Units
Geom File=g01
Flow File=f01
Plan File=p01
Y Axis Title=Elevation
X Axis Title(PF)=Main Channel Distance
X Axis Title(XS)=Station
BEGIN DESCRIPTION:
MDW T 021
END DESCRIPTION:
DSS Export Rating Curves= 0
DSS Export Rating Curve Sorted= 0
DSS Export Volume Flow Curves= 0
DXF OffsetX= 0
DXF OffsetY= 0
DXF ScaleX= 1
DXF ScaleY= 10

--- MDW T 021.p01 (plan) ---

Plan Title=Multiple Run
Short Identifier=Multiple
Geom File=g01
Flow File=f01
Subcritical Flow
K Sum by GR= 0
Std Step Tol= 0.01
Critical Tol= 0.01
Num of Std Step Trials= 20
Max Error Tol= 0.3
Flow Tol Ratio= 0.001
Split Flow NTrial= 30
Split Flow Tol= 0.02
Split Flow Ratio= 0.02
Log Output Level= 0
Friction Slope Method= 1
Unsteady Friction Slope Method= 2
Unsteady Bridges Friction Slope Method= 1
Parabolic Critical Depth
Global Vel Dist=  1 , 1 , 1
Global Log Level= 0
CheckData=True
Encroach Param= -1, 0, 0, 0
BEGIN DESCRIPTION:
Multiple Run
END DESCRIPTION:

--- MDW T 021.f01 (steady flow) ---

Flow Title=Multiple
Number of Profiles=7
Profile Names=10-year,25-year,50-year,1pct_min,100-year,1pct_plu,500-year
River Rch & RM= MDW T 021,Reach-1,17873
     581     796     973     591    1179    2353    1735
River Rch & RM= MDW T 021,Reach-1,13342
     791    1103    1365     838    1673    3338    2519
River Rch & RM= MDW T 021,Reach-1,12995
     880    1231    1527     939    1873    3738    2829
River Rch & RM= MDW T 021,Reach-1,8582
    1127    1597    1998    1239    2471    4931    3793
River Rch & RM= MDW T 021,Reach-1,3829
    1166    1656    2073    1286    2566    5119    3943
River Rch & RM= MDW T 021,Reach-1,2757
    1182    1678    2101    1303    2600    5187    3993
Boundary for River Rch & Prof#=MDW T 021,Reach-1,1
Up Type=0
Dn Type=3
Dn Slope=0.005
Boundary for River Rch & Prof#=MDW T 021,Reach-1,2
Up Type=0
Dn Type=3
Dn Slope=0.005
Boundary for River Rch & Prof#=MDW T 021,Reach-1,3
Up Type=0
Dn Type=3
Dn Slope=0.005
Boundary for River Rch & Prof#=MDW T 021,Reach-1,4
Up Type=0
Dn Type=3
Dn Slope=0.005
Boundary for River Rch & Prof#=MDW T 021,Reach-1,5
Up Type=0
Dn Type=3
Dn Slope=0.005
Boundary for River Rch & Prof#=MDW T 021,Reach-1,6
Up Type=0
Dn Type=3
Dn Slope=0.005
Boundary for River Rch & Prof#=MDW T 021,Reach-1,7
Up Type=0
Dn Type=3
Dn Slope=0.005

--- MDW T 021.g01 (geometry) ---

Geom Title=Existing Conditions

River Reach=MDW T 021,Reach-1
Reach XY= 30
      2284479.00      7116910.00      2284753.19      7115779.45
      2285425.52      7115077.93      2285238.81      7114607.38
      2285909.22      7113960.19      2285865.01      7113375.58
      2286088.80      7113128.15      2286027.40      7112838.85
      2286235.87      7112552.22      2286196.31      7112365.02
      2286424.45      7112256.90      2286484.81      7111785.40
      2286283.21      7111520.18      2286455.31      7111302.82
      2286398.00      7111032.24      2286886.62      7110868.95
      2286991.61      7110506.58      2288046.88      7109372.47
      2287889.60      7108671.25      2288078.93      7108447.27
      2287849.98      7108202.16      2287750.54      7107572.84
      2287901.36      7106625.05      2287803.08      7106309.90
      2288180.45      7106037.55      2288176.68      7105772.44
      2288462.57      7105499.56      2288822.61      7103315.57
      2289237.53      7103342.56      2289179.00      7102960.00

Type RM Length L Ch R = 1,17873,334,334,334
BEGIN DESCRIPTION:
MDW T 021 36.0
END DESCRIPTION:
XS GIS Cut Line= 3
      2284788.64      7116930.63      2284474.59      7116757.93
      2284052.85      7116547.55
#Sta/Elev= 30
  4641.6  893.74  4709.7  891.73  4840.5  886.04  4981.6  885.22  4987.3  884.81
  4992.6  881.52  4992.9  881.02  4996.4  881.02  4996.6  881.52  5003.6  881.83
  5009.2  883.78  5026.0  884.46  5031.6  883.77  5048.4  883.86  5054.0  882.94
  5076.3  883.58  5098.7  882.72  5106.8  884.13  5115.5  884.34  5143.5  884.05
  5233.0  885.42  5255.3  887.01  5272.1  889.89  5277.7  890.01  5316.9  894.42
  5389.6  896.40  5397.4  897.64  5406.4  897.95  5434.3  897.87  5471.3  899.54
#Mann=3,-1,0
  4641.6    0.05       0  4992.6    0.04       0  4996.6    0.05       0
Bank Sta=4992.6,4996.6
Exp/Cntr=0.3,0.1

Type RM Length L Ch R = 1,17539,269,269,269
BEGIN DESCRIPTION:
MDW T 021 35.0
END DESCRIPTION:
XS GIS Cut Line= 3
      2284975.70      7116704.52      2284624.48      7116499.69
      2284183.82      7116306.59
#Sta/Elev= 30
  4598.2  892.90  4641.7  891.19  4673.1  890.49  4687.0  889.59  4694.6  889.67
  4700.4  888.94  4710.1  889.17  4812.1  886.47  4849.1  886.02  4876.6  884.73
  4919.6  883.91  4941.7  882.85  5004.8  882.03  5008.8  879.41  5009.0  878.91
  5012.5  878.91  5012.8  879.41  5021.8  879.46  5032.6  881.87  5120.8  881.69
  5174.5  885.34  5214.3  886.36  5272.8  888.74  5295.3  889.00  5336.6  890.78
  5342.1  890.44  5403.8  893.09  5417.7  892.99  5447.5  894.77  5485.9  895.96
#Mann=3,-1,0
  4598.2    0.05       0  5008.8    0.04       0  5012.8    0.05       0
Bank Sta=5008.8,5012.8
Exp/Cntr=0.3,0.1

Type RM Length L Ch R = 1,17270,287,287,287
BEGIN DESCRIPTION:
Mapping XS 30ca60dc
END DESCRIPTION:
XS GIS Cut Line= 2
      2285042.11      7116354.98      2284345.33      7116150.75
#Sta/Elev= 30
  4621.6  886.09  4666.5  884.86  4687.4  884.88  4697.8  884.15  4731.2  883.16
  4759.4  879.90  4770.7  879.54  4791.6  879.79  4798.0  878.89  4812.4  880.14
  4903.5  879.33  4916.6  878.86  4925.0  877.90  4925.3  877.40  4928.8  877.40
  4929.0  877.90  4936.9  879.01  4942.1  879.10  4958.3  878.84  4968.7  879.26
  4980.7  878.42  5008.9  880.28  5062.5  880.06  5093.8  880.78  5177.1  884.19
  5191.6  884.14  5225.0  885.98  5258.4  886.84  5297.0  888.80  5347.7  890.51
#Mann=3,-1,0
  4621.6    0.05       0  4925.0    0.04       0  4929.0    0.05       0
#XS Ineff=2,0
    0.00 4827.10  885.67 5172.90    0.00  885.67
Permanent Ineff=
       F       F
Bank Sta=4925,4929
Exp/Cntr=0.3,0.1

Type RM Length L Ch R = 1,16983,155,155,155
BEGIN DESCRIPTION:
Mapping XS 03f3f18d
END DESCRIPTION:
XS GIS Cut Line= 2
      2285106.70      7116228.36      2284469.87      7115920.82
#Sta/Elev= 30
  4514.9  885.38  4525.8  884.55  4548.4  883.73  4616.2  882.00  4655.9  881.32
  4667.8  880.26  4684.0  879.64  4723.3  879.23  4745.6  878.60  4774.4  879.03
  4812.2  878.50  4842.3  878.91  4847.8  878.50  4887.5  878.80  4945.4  877.46
  4983.4  877.23  5004.0  875.13  5004.3  874.63  5007.8  874.63  5008.0  875.13
  5023.1  877.31  5028.6  877.75  5067.6  879.79  5073.8  880.43  5119.0  882.55
  5141.6  884.18  5164.2  884.74  5186.8  885.77  5192.4  885.52  5222.1  886.57
#Mann=3,-1,0
  4514.9    0.05       0  5004.0    0.04       0  5008.0    0.05       0
Bank Sta=5004,5008
Exp/Cntr=0.3,0.1

Type RM Length L Ch R = 1,16828,110,110,110
BEGIN DESCRIPTION:
MDW T 021 34.0
END DESCRIPTION:
XS GIS Cut Line= 3
      2285421.78      7115895.88      2284744.15      7115885.11
      2284029.05      7115896.41
#Sta/Elev= 30
  4323.3  889.04  4336.1  889.17  4366.1  886.85  4436.1  884.31  4566.1  881.26
  4726.1  878.32  4766.1  878.45  4776.1  877.74  4806.1  877.23  4886.1  876.82
  4916.2  877.37  4956.2  876.59  4986.2  877.04  4996.1  874.97  5014.2  874.83
  5014.4  874.33  5017.9  874.33  5018.2  874.83  5036.2  877.10  5076.2  878.12
  5116.2  881.55  5256.2  886.18  5326.2  889.96  5466.2  895.64  5506.2  898.07
  5566.2  900.66  5606.2  903.05  5624.0  904.89  5629.0  904.60  5716.2  910.45
#Mann=3,-1,0
  4323.3    0.05       0  5014.2   0.033       0  5018.2    0.05       0
Bank Sta=5014.2,5018.2
Exp/Cntr=0.3,0.1

Type RM Length L Ch R = 1,16718,455,455,455
BEGIN DESCRIPTION:
MDW T 021 33.0
END DESCRIPTION:
XS GIS Cut Line= 3
      2285648.85      7115745.37      2284748.11      7115778.34
      2284025.56      7115780.09
#Sta/Elev= 30
  4104.6  894.37  4124.5  894.55  4174.5  892.16  4274.6  889.68  4363.7  884.27
  4584.8  877.06  4604.8  875.70  4614.8  873.45  4632.8  871.64  4633.1  871.14
  4636.8  871.64  4640.5  872.49  4684.8  873.26  4754.9  873.23  4764.9  872.23
  4804.9  874.46  4875.0  875.52  4895.0  873.43  4917.3  875.34  4945.0  874.31
  4965.0  875.52  4995.0  872.18  5008.0  872.37  5035.1  876.93  5135.1  882.36
  5235.1  885.73  5315.1  890.20  5465.1  896.48  5585.1  903.04  5728.5  912.55
#Mann=3,-1,0
  4104.6    0.05       0  4632.8   0.033       0  4636.8    0.05       0
#XS Ineff=1,-1
 4850.00 5571.00  893.36
Permanent Ineff=
       F
Bank Sta=4632.8,4636.8
Exp/Cntr=0.3,0.1

Type RM Length L Ch R = 1,16263,318,318,318
BEGIN DESCRIPTION:
MDW T 021 32.0
END DESCRIPTION:
XS GIS Cut Line= 3
      2285657.51      7115665.50      2285080.41      7115476.14
      2284318.99      7115233.22
#Sta/Elev= 30
  4396.2  893.08  4430.7  892.81  4468.3  890.35  4542.0  887.79  4595.1  881.86
  4621.6  880.34  4678.8  879.32  4763.0  875.67  4826.1  874.12  4849.7  871.30
  4857.7  869.44  4868.2  870.10  4876.2  872.35  4971.7  872.12  4994.5  870.46
  4999.7  867.49  4999.9  866.99  5003.7  867.49  5008.8  867.57  5015.5  871.48
  5026.0  872.55  5207.2  871.42  5239.4  874.35  5257.0  877.21  5278.0  878.37
  5373.5  882.22  5487.9  888.74  5561.4  891.32  5750.3  900.81  5802.8  904.19
#Mann=3,-1,0
  4396.2    0.05       0  4999.7   0.033       0  5003.7    0.05       0
Bank Sta=4999.7,5003.7
Exp/Cntr=0.3,0.1

Type RM Length L Ch R = 1,15945,212,212,212
BEGIN DESCRIPTION:
MDW T 021 31.0
END DESCRIPTION:
XS GIS Cut Line= 3
      2285697.45      7115573.49      2285278.13      7115244.64
      2284478.72      7114809.62
#Sta/Elev= 30
  4460.3  891.01  4560.7  887.91  4668.3  878.24  4732.4  877.14  4753.3  875.13
  4761.4  875.52  4767.7  874.44  4796.6  874.32  4817.4  872.88  4839.6  873.18
  4852.7  871.88  4889.7  872.76  4960.3  870.55  4989.2  868.52  4992.9  865.93
  5001.6  865.71  5001.8  865.21  5005.6  865.71  5011.3  869.58  5017.0  869.98
  5151.6  869.55  5333.7  873.73  5387.5  880.38  5447.3  881.09  5496.7  882.89
  5681.9  892.16  5719.9  892.56  5807.3  897.61  5880.2  898.88  5903.3  900.37
#Mann=3,-1,0
  4460.3    0.05       0  5001.6   0.033       0  5005.6    0.05       0
Bank Sta=5001.6,5005.6
Exp/Cntr=0.3,0.1

Type RM Length L Ch R = 1,15733,313,313,313
BEGIN DESCRIPTION:
Mapping XS ff091364
END DESCRIPTION:
XS GIS Cut Line= 3
      2285675.26      7115333.13      2285270.30      7114950.68
      2284985.46      7114822.89
#Sta/Elev= 30
  4646.4  879.56  4653.2  880.23  4660.1  880.09  4674.2  878.17  4716.7  876.37
  4730.9  876.15  4737.7  876.81  4751.9  875.11  4815.8  872.39  4836.9  870.39
  4844.1  868.46  4851.0  867.76  4978.4  868.43  4983.3  865.80  4983.6  865.30
  4987.1  865.30  4987.3  865.80  4999.5  865.97  5006.8  866.82  5013.6  868.44
  5020.9  867.63  5084.4  868.15  5134.2  869.68  5169.4  868.97  5200.9  870.06
  5237.0  870.52  5288.8  872.42  5294.3  872.12  5380.2  875.26  5515.6  878.84
#Mann=3,-1,0
  4646.4    0.05       0  4983.3   0.033       0  4987.3    0.05       0
Bank Sta=4983.3,4987.3
Exp/Cntr=0.3,0.1

Type RM Length L Ch R = 1,15420,268,268,268
BEGIN DESCRIPTION:
Mapping XS 922134d2
END DESCRIPTION:
XS GIS Cut Line= 2
      2285790.97      7114832.60      2285073.32      7114809.95
#Sta/Elev= 30
  4622.4  868.47  4664.4  867.83  4714.4  868.07  4764.4  866.78  4784.4  866.56
  4814.5  866.92  4824.5  865.97  4884.5  866.20  4894.5  866.60  4904.5  866.07
  4964.5  865.83  4974.5  865.67  4984.5  864.21  4992.6  863.68  4992.8  863.18
  4996.3  863.18  4996.6  863.68  5004.6  864.95  5034.6  865.74  5054.6  865.63
  5084.6  867.29  5094.6  868.20  5114.6  868.88  5124.6  869.64  5144.6  870.46
  5180.0  871.46  5194.6  871.55  5244.7  873.28  5314.7  874.98  5340.4  875.91
#Mann=3,-1,0
  4622.4    0.05       0  4992.6   0.033       0  4996.6    0.05       0
Bank Sta=4992.6,4996.6
Exp/Cntr=0.3,0.1

Type RM Length L Ch R = 1,15152,317,317,317
BEGIN DESCRIPTION:
Mapping XS db193223
END DESCRIPTION:
XS GIS Cut Line= 2
      2285751.41      7114632.22      2284967.28      7114642.67
#Sta/Elev= 30
  4494.5  865.78  4536.9  865.58  4576.9  866.13  4606.9  866.05  4656.9  867.12
  4666.9  866.46  4686.9  865.94  4726.9  865.44  4756.9  865.39  4766.9  865.82
  4786.9  865.38  4796.9  865.80  4856.9  864.73  4876.9  865.17  4886.9  864.94
  4956.9  865.21  4966.9  864.45  4987.0  863.71  5005.0  862.21  5005.2  861.71
  5008.7  861.71  5009.0  862.21  5017.0  864.66  5037.0  868.22  5047.0  871.15
  5097.0  873.66  5167.0  876.15  5177.0  876.95  5187.0  877.10  5278.7  881.73
#Mann=3,-1,0
  4494.5    0.05       0  5005.0   0.033       0  5009.0    0.05       0
Bank Sta=5005,5009
Exp/Cntr=0.3,0.1

Type RM Length L Ch R = 1,14835,241,241,241
BEGIN DESCRIPTION:
Mapping XS 681a3260
END DESCRIPTION:
XS GIS Cut Line= 2
      2285806.39      7114599.01      2285093.59      7114277.88
#Sta/Elev= 30
  4571.0  865.61  4657.6  864.76  4765.6  864.95  4809.4  866.24  4864.3  864.76
  4886.2  863.21  4930.1  864.10  4952.0  863.84  4963.0  861.00  4984.9  860.51
  4992.5  861.82  4996.0  859.20  4996.3  858.70  4999.8  858.70  5000.0  859.20
  5006.9  860.42  5015.7  859.87  5021.1  860.40  5028.8  862.92  5038.8  863.08
  5044.3  862.27  5067.4  865.13  5136.9  867.85  5165.5  868.23  5211.8  870.33
  5234.9  871.03  5240.4  870.55  5258.0  871.56  5263.5  871.26  5352.8  873.93
#Mann=3,-1,0
  4571.0    0.05       0  4996.0   0.033       0  5000.0    0.05       0
Bank Sta=4996,5000
Exp/Cntr=0.3,0.1

Type RM Length L Ch R = 1,14594,147,147,147
BEGIN DESCRIPTION:
MDW T 021 28.0
END DESCRIPTION:
XS GIS Cut Line= 3
      2285869.80      7114550.40      2285580.83      7114248.97
      2285117.23      7113897.24
#Sta/Elev= 30
  4550.6  866.06  4685.9  863.45  4820.2  863.76  4947.6  862.76  4971.5  863.57
  4983.0  862.81  4990.3  857.27  4994.6  856.52  4994.8  856.02  4998.6  856.52
  5004.8  856.98  5011.1  860.27  5019.4  862.22  5040.2  860.87  5046.5  861.82
  5061.0  862.05  5146.3  861.70  5160.9  861.02  5210.8  861.55  5233.6  863.33
  5239.9  864.92  5254.4  865.72  5283.5  866.79  5289.8  865.82  5296.8  867.43
  5310.6  867.31  5318.9  868.11  5389.7  870.15  5404.2  871.42  5550.1  877.23
#Mann=3,-1,0
  4550.6    0.05       0  4994.6   0.033       0  4998.6    0.05       0
Bank Sta=4994.6,4998.6
Exp/Cntr=0.3,0.1

Type RM Length L Ch R = 1,14447,480,480,480
BEGIN DESCRIPTION:
Mapping XS e8f30b1c
END DESCRIPTION:
XS GIS Cut Line= 4
      2285842.36      7114490.24      2285608.77      7114038.64
      2285532.10      7113840.49      2285267.80      7113840.48
#Sta/Elev= 30
  4578.7  864.66  4640.7  863.29  4773.5  863.13  4894.2  862.08  4900.7  861.47
  4983.7  859.94  4989.3  857.74  5009.4  857.06  5009.7  856.56  5013.2  856.56
  5013.4  857.06  5033.6  860.17  5083.6  859.47  5131.0  860.09  5155.6  859.23
  5160.9  859.88  5180.2  858.78  5203.6  858.84  5270.0  859.69  5297.2  861.46
  5312.7  861.14  5322.7  858.94  5332.7  858.27  5342.7  858.94  5362.7  858.51
  5372.7  860.13  5382.7  862.70  5392.7  863.65  5492.7  867.30  5563.9  871.26
#Mann=3,-1,0
  4578.7    0.05       0  5009.4   0.033       0  5013.4    0.05       0
Bank Sta=5009.4,5013.4
Exp/Cntr=0.3,0.1

Type RM Length L Ch R = 1,13967,112,112,112
BEGIN DESCRIPTION:
Mapping XS 34ef4f79
END DESCRIPTION:
XS GIS Cut Line= 3
      2286183.52      7113787.19      2285543.28      7113814.63
      2285327.03      7113817.69
#Sta/Elev= 30
  4758.8  859.58  4843.4  858.12  4923.5  857.52  4939.9  856.83  4993.5  857.27
  5003.5  855.35  5011.6  855.19  5011.8  854.69  5015.3  854.69  5015.6  855.19
  5033.6  856.59  5053.6  855.55  5073.6  856.87  5093.6  856.65  5123.7  857.65
  5171.7  857.51  5176.7  858.34  5183.7  858.42  5293.8  858.27  5313.8  858.94
  5343.9  858.87  5373.9  860.28  5383.9  861.42  5422.3  862.23  5433.9  861.70
  5453.9  859.68  5463.9  860.07  5473.9  861.95  5483.9  862.58  5615.9  868.20
#Mann=3,-1,0
  4758.8    0.05       0  5011.6   0.033       0  5015.6    0.05       0
Bank Sta=5011.6,5015.6
Exp/Cntr=0.3,0.1

Type RM Length L Ch R = 1,13855,189,189,189
BEGIN DESCRIPTION:
Mapping XS 16a9ebd4
END DESCRIPTION:
XS GIS Cut Line= 2
      2286158.13      7113696.04      2285439.13      7113740.88
#Sta/Elev= 30
  4775.3  858.78  4844.6  858.56  4864.6  858.11  4904.7  857.66  4934.7  856.47
  4964.8  856.11  4974.8  856.23  4982.8  855.88  4983.1  855.38  4986.6  855.38
  4986.8  855.88  5004.9  856.81  5065.0  857.81  5105.1  857.65  5155.2  857.95
  5165.2  857.72  5185.2  857.87  5195.2  857.48  5205.3  857.43  5215.3  857.77
  5235.3  857.35  5245.5  857.88  5265.4  858.02  5305.5  858.79  5365.6  860.31
  5400.9  861.51  5425.7  862.04  5475.8  863.56  5485.8  863.68  5495.7  864.13
#Mann=3,-1,0
  4775.3    0.05       0  4982.8   0.033       0  4986.8    0.05       0
Bank Sta=4982.8,4986.8
Exp/Cntr=0.3,0.1

Type RM Length L Ch R = 1,13666,324,324,324
BEGIN DESCRIPTION:
Mapping XS a87e9c59
END DESCRIPTION:
XS GIS Cut Line= 3
      2286204.80      7113643.53      2285989.31      7113543.73
      2285313.42      7113485.16
#Sta/Elev= 30
  4655.1  860.06  4676.7  859.67  4683.5  859.90  4699.6  859.39  4705.6  857.96
  4716.6  857.31  4728.1  857.09  4814.2  857.61  4923.0  857.62  4943.1  857.05
  4963.2  855.20  4973.2  855.09  4983.2  854.23  4988.9  851.35  4989.2  850.85
  4992.7  850.85  4992.9  851.35  4996.0  852.86  5003.3  852.06  5013.3  852.70
  5023.4  855.10  5053.5  854.78  5143.8  856.23  5173.9  855.64  5227.2  856.60
  5324.5  859.62  5404.8  863.11  5445.0  865.36  5555.4  870.73  5571.0  871.84
#Mann=3,-1,0
  4655.1    0.05       0  4988.9   0.033       0  4992.9    0.05       0
Bank Sta=4988.9,4992.9
Exp/Cntr=0.3,0.1

Type RM Length L Ch R = 1,13342,347,347,347
BEGIN DESCRIPTION:
MDW T 021 25.0
END DESCRIPTION:
XS GIS Cut Line= 3
      2287054.46      7113759.05      2285980.70      7113270.70
      2285087.41      7113042.02
#Sta/Elev= 30
  3825.6  885.11  3853.6  885.22  3910.9  882.00  3980.1  880.97  4008.7  878.97
  4031.7  879.31  4049.3  878.08  4054.8  879.08  4077.9  878.89  4198.7  874.58
  4238.1  873.08  4314.0  868.36  4584.2  857.37  4681.9  855.01  4743.4  855.02
  4900.5  852.48  4923.5  853.17  4985.1  852.63  4990.7  849.88  4991.0  849.38
  4994.7  849.88  5003.4  851.31  5017.3  852.03  5311.0  857.28  5409.5  861.99
  5461.1  863.26  5550.6  868.52  5646.9  870.05  5673.1  872.65  5927.3  883.67
#Mann=3,-1,0
  3825.6    0.05       0  4990.7    0.04       0  4994.7    0.05       0
Bank Sta=4990.7,4994.7
Exp/Cntr=0.3,0.1

Type RM Length L Ch R = 1,12995,508,508,508
BEGIN DESCRIPTION:
MDW T 021 24.0
END DESCRIPTION:
XS GIS Cut Line= 3
      2286878.96      7113359.98      2286079.44      7112966.32
      2285278.95      7112859.99
#Sta/Elev= 30
  4106.9  876.27  4160.2  872.16  4205.2  869.68  4368.0  863.43  4502.8  859.26
  4615.1  856.44  4755.5  853.74  4862.2  852.60  4912.7  851.00  4957.7  850.50
  4965.1  849.15  4985.0  848.66  4985.6  848.16  4989.3  848.16  4989.8  848.66
  5000.8  848.85  5005.8  849.97  5010.9  848.87  5018.7  850.53  5069.1  849.45
  5119.6  850.20  5180.1  851.94  5301.2  857.83  5331.4  858.41  5387.4  860.53
  5460.6  862.60  5465.7  862.32  5644.1  869.43  5695.6  871.01  5805.6  875.82
#Mann=3,-1,0
  4106.9    0.05       0  4985.0    0.04       0  4989.8    0.05       0
Bank Sta=4985,4989.8
Exp/Cntr=0.3,0.1

Type RM Length L Ch R = 1,12487,309,309,309
BEGIN DESCRIPTION:
MDW T 021 23.0
END DESCRIPTION:
XS GIS Cut Line= 3
      2287151.91      7112910.20      2286227.07      7112554.02
      2285395.39      7112285.19
#Sta/Elev= 30
  4016.1  873.89  4087.5  873.46  4112.2  870.83  4233.5  866.43  4244.3  866.96
  4297.8  865.19  4512.2  857.09  4723.7  851.49  4868.2  848.80  4962.2  848.33
  4972.1  848.04  4991.9  845.43  4992.5  844.93  4996.8  845.43  5026.1  847.78
  5057.7  847.55  5078.7  849.67  5135.3  849.74  5231.3  852.94  5278.4  853.37
  5351.9  855.54  5373.0  855.12  5487.5  858.62  5626.1  861.56  5684.9  864.18
  5845.0  865.21  5856.4  865.61  5866.9  868.57  5876.7  870.47  5881.2  870.47
#Mann=3,-1,0
  4016.1    0.05       0  4991.9    0.04       0  4996.8    0.05       0
Bank Sta=4991.9,4996.8
Exp/Cntr=0.3,0.1

Type RM Length L Ch R = 1,12178,486,486,486
BEGIN DESCRIPTION:
MDW T 021 22.0
END DESCRIPTION:
XS GIS Cut Line= 3
      2287164.46      7112648.46      2286272.97      7112311.89
      2285426.62      7111979.19
#Sta/Elev= 30
  4050.7  870.68  4067.2  869.28  4201.5  864.45  4462.7  856.38  4505.5  856.70
  4517.5  855.57  4644.4  852.10  4751.3  847.40  4847.5  846.59  4890.3  848.15
  4901.0  846.06  4913.4  845.58  4975.8  846.09  4986.5  845.41  4990.9  843.35
  4991.5  842.85  4995.8  843.35  5008.4  844.15  5017.8  845.88  5023.2  845.60
  5029.4  847.22  5269.8  850.26  5299.6  851.66  5378.2  852.95  5402.6  854.83
  5523.6  856.22  5588.1  857.97  5727.8  862.94  5856.7  870.12  5913.0  871.87
#Mann=3,-1,0
  4050.7    0.05       0  4990.9    0.04       0  4995.8    0.05       0
Bank Sta=4990.9,4995.8
Exp/Cntr=0.3,0.1

Type RM Length L Ch R = 1,11692,373,373,373
BEGIN DESCRIPTION:
MDW T 021 21.0
END DESCRIPTION:
XS GIS Cut Line= 3
      2287338.05      7112384.57      2286399.08      7111990.04
      2285518.67      7111686.67
#Sta/Elev= 30
  3985.4  869.77  4233.8  862.52  4331.5  858.14  4515.9  853.88  4591.8  851.01
  4635.2  850.61  4806.8  844.91  4971.4  843.90  4982.3  843.48  4989.4  841.06
  4994.8  841.77  4998.8  841.01  4999.4  840.51  5003.7  841.01  5014.3  843.03
  5035.7  844.21  5201.6  846.21  5232.8  846.30  5238.1  845.35  5405.9  849.00
  5437.6  850.76  5477.2  854.59  5490.5  853.72  5539.6  857.10  5690.4  863.86
  5726.9  866.15  5752.9  870.00  5765.5  870.84  5883.0  871.43  5935.1  873.72
#Mann=3,-1,0
  3985.4    0.05       0  4998.8    0.04       0  5003.7    0.05       0
Bank Sta=4998.8,5003.7
Exp/Cntr=0.3,0.1

Type RM Length L Ch R = 1,11319,288,288,288
BEGIN DESCRIPTION:
Mapping XS 43cb9217
END DESCRIPTION:
XS GIS Cut Line= 2
      2286789.92      7111658.25      2285866.19      7111745.11
#Sta/Elev= 30
  4633.6  847.01  4765.1  846.20  4875.6  843.21  4966.0  843.06  4976.0  842.46
  4986.1  839.44  5003.7  838.76  5004.3  838.26  5008.1  838.26  5008.7  838.76
  5016.2  841.79  5028.7  842.64  5046.3  841.72  5076.5  841.67  5096.6  842.66
  5137.4  842.61  5146.8  843.37  5227.1  843.54  5241.0  844.26  5287.4  844.68
  5337.6  846.40  5418.0  850.13  5448.1  854.99  5453.3  853.96  5458.3  854.78
  5468.2  853.18  5488.3  855.35  5508.4  856.51  5556.9  858.78  5561.4  858.35
#Mann=3,-1,0
  4633.6    0.05       0  5003.7    0.04       0  5008.7    0.05       0
Bank Sta=5003.7,5008.7
Exp/Cntr=0.3,0.1

Type RM Length L Ch R = 1,11031,209,209,209
BEGIN DESCRIPTION:
Mapping XS a028791e
END DESCRIPTION:
XS GIS Cut Line= 2
      2286752.33      7111481.27      2286042.24      7111463.88
#Sta/Elev= 30
  4543.5  845.07  4596.8  844.98  4626.9  844.29  4736.9  843.60  4756.9  842.88
  4776.9  843.08  4806.9  840.66  4836.9  840.14  4866.9  840.25  4886.9  841.22
  4926.9  840.55  4977.0  840.40  4987.0  838.81  4994.4  837.14  4995.1  836.64
  4998.9  836.64  4999.5  837.14  5007.0  838.18  5017.0  841.77  5067.0  841.41
  5087.0  842.04  5097.0  841.87  5187.0  843.55  5197.0  844.72  5205.1  846.58
  5210.1  846.99  5217.0  845.77  5237.0  846.46  5247.0  848.06  5253.8  849.66
#Mann=3,-1,0
  4543.5    0.05       0  4994.4    0.04       0  4999.5    0.05       0
Bank Sta=4994.4,4999.5
Exp/Cntr=0.3,0.1

Type RM Length L Ch R = 1,10822,337,337,337
BEGIN DESCRIPTION:
Mapping XS fe252512
END DESCRIPTION:
XS GIS Cut Line= 4
      2286734.27      7111403.90      2286419.28      7111326.82
      2286288.14      7111349.58      2286109.81      7111330.83
#Sta/Elev= 30
  4699.2  844.06  4838.5  842.72  4869.3  841.86  4900.0  841.88  4910.5  841.51
  4920.8  840.45  4946.8  839.63  4982.6  839.73  4988.4  837.04  4991.0  837.04
  4991.6  836.54  4995.4  836.54  4996.1  837.04  5003.2  837.12  5013.5  838.96
  5033.9  839.02  5054.2  839.89  5075.5  839.80  5115.1  841.07  5175.8  841.30
  5195.6  841.23  5200.7  840.82  5226.1  841.16  5246.2  842.52  5256.3  844.57
  5276.4  845.09  5293.7  843.39  5316.6  845.34  5326.7  844.47  5335.9  844.80
#Mann=3,-1,0
  4699.2    0.05       0  4991.0    0.04       0  4996.1    0.05       0
Bank Sta=4991,4996.1
Exp/Cntr=0.3,0.1

Type RM Length L Ch R = 1,10485,284,284,284
BEGIN DESCRIPTION:
Mapping XS 47e06ace
END DESCRIPTION:
XS GIS Cut Line= 3
      2286726.96      7111254.69      2286606.82      7111184.23
      2286318.29      7110950.82
#Sta/Elev= 30
  4604.1  841.95  4685.6  840.90  4707.1  840.17  4717.0  840.53  4742.6  839.90
  4766.3  840.37  4808.5  838.41  4822.9  838.39  4837.3  839.04  4858.1  837.59
  4901.3  837.77  4915.6  839.04  4922.1  838.38  4930.0  839.84  4936.4  838.67
  4944.4  838.64  4950.8  837.70  4958.8  838.42  4965.2  837.77  4994.0  837.53
  5000.4  837.05  5012.2  834.82  5012.9  834.32  5016.7  834.32  5017.3  834.82
  5022.7  837.21  5036.4  839.14  5072.3  840.40  5086.7  842.05  5114.5  843.61
#Mann=3,-1,0
  4604.1    0.05       0  5012.2    0.04       0  5017.3    0.05       0
Bank Sta=5012.2,5017.3
Exp/Cntr=0.3,0.1

Type RM Length L Ch R = 1,10201,292,292,292
BEGIN DESCRIPTION:
Mapping XS a0591341
END DESCRIPTION:
XS GIS Cut Line= 3
      2286730.75      7111121.90      2286582.59      7110939.27
      2286415.18      7110895.15
#Sta/Elev= 30
  4874.2  840.34  4884.0  839.73  4912.7  840.32  4933.6  838.22  4941.0  838.19
  4947.9  837.14  4954.4  836.97  4962.3  835.53  4976.7  834.95  4983.1  835.17
  4991.1  833.77  4996.0  834.49  5005.4  832.47  5009.3  830.50  5010.0  830.00
  5013.8  830.00  5014.5  830.50  5018.3  833.80  5032.7  832.72  5040.6  835.76
  5047.1  834.83  5055.0  836.23  5069.4  836.23  5096.6  837.63  5133.8  837.41
  5226.8  838.60  5243.1  839.06  5257.9  840.29  5268.2  840.25  5282.5  841.00
#Mann=3,-1,0
  4874.2    0.05       0  5009.3    0.04       0  5014.5    0.05       0
Bank Sta=5009.3,5014.5
Exp/Cntr=0.3,0.1

Type RM Length L Ch R = 1,9909,101,101,101
BEGIN DESCRIPTION:
Mapping XS 354fb0fb
END DESCRIPTION:
XS GIS Cut Line= 2
      2287060.70      7110850.60      2286522.54      7110897.49
#Sta/Elev= 30
  4827.5  838.64  4859.3  837.94  4876.3  837.09  4881.3  837.62  4929.6  836.76
  4939.6  836.34  4949.7  836.36  4959.7  835.69  4969.7  834.53  4979.8  831.01
  4986.5  830.63  4987.2  830.13  4991.0  830.13  4991.7  830.63  5009.9  831.63
  5019.9  831.48  5040.0  833.42  5100.2  834.92  5120.3  834.87  5130.3  835.34
  5140.4  835.27  5150.4  836.13  5210.6  835.12  5219.7  835.20  5224.7  834.85
  5260.8  835.70  5311.0  836.44  5337.5  837.21  5342.6  837.08  5367.7  837.89
#Mann=3,-1,0
  4827.5    0.05       0  4986.5    0.04       0  4991.7    0.05       0
Bank Sta=4986.5,4991.7
Exp/Cntr=0.3,0.1

Type RM Length L Ch R = 1,9808,199,199,199
BEGIN DESCRIPTION:
Mapping XS a54acd95
END DESCRIPTION:
XS GIS Cut Line= 2
      2287160.37      7110756.78      2286462.57      7110820.48
#Sta/Elev= 30
  4775.1  837.24  4863.7  835.61  4868.7  835.96  4876.9  835.76  4886.9  835.99
  4907.0  835.14  4957.2  834.32  4967.3  833.04  4973.9  831.40  4978.9  831.76
  4987.3  831.00  4994.8  829.17  4995.5  828.67  4999.3  828.67  5000.0  829.17
  5017.5  831.71  5037.6  832.57  5047.6  832.50  5084.1  833.18  5107.8  833.27
  5127.9  833.74  5199.4  834.63  5208.3  835.23  5288.6  836.53  5348.8  837.96
  5368.9  838.08  5409.1  839.36  5414.8  839.73  5419.8  839.49  5475.8  841.00
#Mann=3,-1,0
  4775.1    0.05       0  4994.8    0.04       0  5000.0    0.05       0
Bank Sta=4994.8,5000
Exp/Cntr=0.3,0.1

Type RM Length L Ch R = 1,9609,262,262,262
BEGIN DESCRIPTION:
Mapping XS 2170054f
END DESCRIPTION:
XS GIS Cut Line= 2
      2287150.91      7110708.63      2286681.99      7110423.51
#Sta/Elev= 30
  4763.3  835.51  4770.8  835.21  4786.3  834.99  4800.7  834.38  4844.4  833.76
  4859.2  833.28  4887.1  832.93  4945.2  832.77  4982.0  832.16  4987.9  830.56
  4997.5  829.12  5003.4  828.74  5008.7  828.03  5009.4  827.53  5013.2  827.53
  5013.9  828.03  5018.8  829.30  5024.7  830.19  5069.8  831.40  5092.4  832.88
  5135.1  836.15  5140.9  836.06  5171.9  836.87  5199.1  838.04  5208.7  838.20
  5214.6  838.64  5288.2  840.67  5294.0  841.05  5303.6  841.24  5312.1  841.84
#Mann=3,-1,0
  4763.3    0.05       0  5008.7    0.04       0  5013.9    0.05       0
Bank Sta=5008.7,5013.9
Exp/Cntr=0.3,0.1

Type RM Length L Ch R = 1,9347,287,287,287
BEGIN DESCRIPTION:
Mapping XS 53b60daa
END DESCRIPTION:
XS GIS Cut Line= 2
      2287256.38      7110649.98      2287001.03      7110187.72
#Sta/Elev= 30
  4693.7  834.99  4750.8  833.30  4786.1  832.68  4839.9  832.29  4853.6  831.77
  4883.5  831.40  4910.9  831.49  4921.3  831.30  4927.0  831.48  4956.4  830.93
  4964.8  830.45  4979.3  828.75  4986.6  827.80  4992.3  826.32  4999.5  826.12
  5000.2  825.62  5004.0  825.62  5004.8  826.12  5008.3  827.94  5014.1  829.31
  5051.9  829.69  5059.3  829.45  5073.6  830.70  5082.1  831.05  5095.4  832.97
  5105.0  833.40  5139.2  834.12  5149.3  834.06  5171.0  835.16  5221.8  836.19
#Mann=3,-1,0
  4693.7    0.05       0  4999.5    0.04       0  5004.8    0.05       0
Bank Sta=4999.5,5004.8
Exp/Cntr=0.3,0.1

Type RM Length L Ch R = 1,9060,151,151,151
BEGIN DESCRIPTION:
Mapping XS f79a7a34
END DESCRIPTION:
XS GIS Cut Line= 2
      2287409.55      7110402.15      2287222.30      7109973.35
#Sta/Elev= 30
  4759.7  832.44  4822.8  830.74  4828.3  830.85  4846.2  830.36  4851.7  830.56
  4921.9  829.39  4936.6  829.93  4958.5  830.01  4968.7  829.27  4974.1  827.43
  4980.3  825.98  4991.2  824.86  5000.4  824.70  5001.1  824.20  5004.9  824.20
  5005.7  824.70  5013.0  824.72  5021.0  825.19  5026.4  827.64  5049.8  828.45
  5073.2  828.63  5102.1  830.12  5120.0  830.32  5143.4  830.98  5148.9  831.43
  5177.8  832.30  5187.6  832.40  5201.2  833.69  5219.1  833.77  5227.6  834.11
#Mann=3,-1,0
  4759.7    0.05       0  5000.4    0.04       0  5005.7    0.05       0
Bank Sta=5000.4,5005.7
Exp/Cntr=0.3,0.1

Type RM Length L Ch R = 1,8909,327,327,327
BEGIN DESCRIPTION:
Mapping XS 1b928eab
END DESCRIPTION:
XS GIS Cut Line= 2
      2287541.76      7110283.95      2287294.60      7109876.32
#Sta/Elev= 30
  4744.0  831.39  4749.2  831.39  4778.1  830.11  4793.5  829.89  4830.4  828.75
  4842.2  828.87  4873.0  828.21  4915.7  828.87  4931.2  828.34  4959.1  828.21
  4968.0  827.83  4982.5  825.82  4989.4  824.46  4992.6  824.20  4993.3  823.70
  4997.1  823.70  4997.9  824.20  5010.7  824.28  5026.2  825.69  5032.1  827.14
  5076.1  829.25  5084.4  829.22  5090.2  829.67  5121.2  829.81  5142.6  830.54
  5148.4  831.18  5163.9  831.17  5185.2  831.64  5193.0  832.18  5220.7  832.50
#Mann=3,-1,0
  4744.0    0.05       0  4992.6    0.04       0  4997.9    0.05       0
Bank Sta=4992.6,4997.9
Exp/Cntr=0.3,0.1

Type RM Length L Ch R = 1,8582,206,206,206
BEGIN DESCRIPTION:
Mapping XS a124624f
END DESCRIPTION:
XS GIS Cut Line= 4
      2287676.21      7110211.16      2287739.51      7110010.44
      2287587.43      7109741.60      2287296.17      7109665.80
#Sta/Elev= 30
  4628.5  832.99  4649.9  832.24  4655.2  832.84  4719.9  830.76  4725.1  831.20
  4776.5  828.17  4808.0  827.79  4828.9  829.01  4842.1  828.68  4906.9  826.12
  4912.6  825.34  4919.9  822.26  4990.7  822.19  4991.5  821.69  4996.1  822.19
  5015.1  822.41  5023.3  823.65  5036.7  824.09  5095.9  824.94  5103.7  827.36
  5111.8  826.75  5117.6  832.11  5133.5  832.55  5145.9  832.45  5156.5  831.29
  5352.9  831.31  5411.0  831.62  5416.1  831.78  5425.2  833.54  5448.8  832.06
#Mann=3,-1,0
  4628.5    0.05       0  4990.7    0.04       0  4996.1    0.05       0
Bank Sta=4990.7,4996.1
Exp/Cntr=0.3,0.1

Type RM Length L Ch R = 1,8376,245,245,245
BEGIN DESCRIPTION:
Mapping XS 16d94aea
END DESCRIPTION:
XS GIS Cut Line= 2
      2288169.34      7109948.75      2287376.67      7109499.95
#Sta/Elev= 30
  4545.9  844.79  4596.1  842.76  4661.2  838.18  4764.6  832.18  4832.7  829.25
  4838.5  828.78  4845.1  826.63  4854.4  822.60  4876.0  822.88  5072.2  822.40
  5073.0  821.90  5076.9  821.90  5077.6  822.40  5086.7  822.43  5096.8  824.26
  5140.1  825.07  5145.9  826.16  5161.7  832.54  5167.5  832.73  5189.8  832.83
  5199.3  832.08  5220.9  832.28  5226.7  831.29  5235.8  831.51  5258.5  831.04
  5280.1  831.55  5316.2  830.86  5323.4  831.56  5350.8  830.96  5456.8  831.43
#Mann=3,-1,0
  4545.9    0.05       0  5072.2    0.04       0  5077.6    0.05       0
Bank Sta=5072.2,5077.6
Exp/Cntr=0.3,0.1

Type RM Length L Ch R = 1,8131,362,362,362
BEGIN DESCRIPTION:
Mapping XS 1ef4ddb8
END DESCRIPTION:
XS GIS Cut Line= 2
      2288242.19      7109668.25      2287346.81      7109294.91
#Sta/Elev= 30
  4661.7  847.83  4708.5  847.55  4718.0  847.00  4723.4  846.36  4741.0  841.92
  4747.3  839.59  4752.7  838.87  4771.1  834.50  4806.0  831.35  4871.0  826.84
  4892.7  824.91  4901.1  822.94  4906.5  823.28  5063.3  822.27  5064.1  821.77
  5068.0  821.77  5068.7  822.27  5184.8  822.65  5196.0  823.98  5237.9  824.82
  5243.3  825.90  5250.2  829.75  5261.1  831.97  5267.1  832.23  5320.2  831.33
  5434.4  831.69  5596.9  831.10  5609.4  832.16  5618.6  832.29  5631.8  831.26
#Mann=3,-1,0
  4661.7    0.05       0  5063.3    0.04       0  5068.7    0.05       0
Bank Sta=5063.3,5068.7
Exp/Cntr=0.3,0.1

Type RM Length L Ch R = 1,7769,107,107,107
BEGIN DESCRIPTION:
Mapping XS ca30459f
END DESCRIPTION:
XS GIS Cut Line= 2
      2288314.72      7109219.00      2287215.84      7109226.27
#Sta/Elev= 30
  4684.4  838.61  4690.1  837.18  4710.1  834.89  4730.1  833.83  4750.1  831.60
  4800.1  827.85  4830.1  826.82  4840.1  825.95  4850.1  822.33  4970.1  822.78
  5007.0  817.62  5008.1  817.12  5012.2  817.12  5013.2  817.62  5030.1  819.53
  5070.1  825.63  5120.1  823.94  5150.1  823.52  5200.1  824.80  5230.1  826.28
  5270.1  827.13  5320.1  826.73  5380.1  827.87  5490.1  828.37  5620.1  829.95
  5630.1  829.54  5710.1  831.35  5730.1  831.07  5740.1  831.62  5783.3  831.75
#Mann=3,-1,0
  4684.4    0.05       0  5007.0   0.033       0  5013.2    0.05       0
#XS Ineff=2,0
       0                 5063.00    0.00  831.48
Permanent Ineff=
       F       F
Bank Sta=5007,5013.2
Exp/Cntr=0.3,0.1

Type RM Length L Ch R = 1,7662,136,136,136
BEGIN DESCRIPTION:
Mapping XS bdd37fa5
END DESCRIPTION:
XS GIS Cut Line= 2
      2288341.88      7109117.94      2287232.43      7109106.92
#Sta/Elev= 30
  4654.4  837.49  4658.3  837.49  4667.3  835.70  4737.3  830.39  4827.3  825.03
  4857.3  823.61  4907.3  823.71  4946.4  822.83  4977.3  818.55  5004.2  815.99
  5005.2  815.49  5009.3  815.49  5010.4  815.99  5017.3  816.98  5027.3  820.16
  5037.3  820.93  5047.3  821.30  5097.3  821.48  5117.3  822.07  5157.3  824.41
  5267.3  826.19  5297.3  825.99  5317.3  826.26  5347.3  827.21  5357.3  827.18
  5387.3  828.83  5547.3  829.69  5637.3  829.72  5647.3  830.40  5763.9  831.46
#Mann=3,-1,0
  4654.4    0.05       0  5004.2   0.033       0  5010.4    0.05       0
Bank Sta=5004.2,5010.4
Exp/Cntr=0.3,0.1

Type RM Length L Ch R = 1,7526,365,365,365
BEGIN DESCRIPTION:
MDW T 021 12.0
END DESCRIPTION:
XS GIS Cut Line= 3
      2288442.89      7109013.30      2287931.91      7109003.97
      2286399.57      7108957.74
#Sta/Elev= 30
  4493.6  840.93  4537.5  840.33  4577.5  838.78  4597.5  833.15  4677.5  826.96
  4757.5  823.38  4877.6  820.64  4927.6  818.12  4950.3  817.90  4994.5  814.65
  4995.5  814.15  5000.7  814.65  5057.6  821.78  5077.6  822.82  5177.7  823.38
  5217.7  824.74  5267.7  824.48  5357.7  825.56  5467.8  827.67  5477.8  828.53
  5517.8  828.41  5527.8  829.00  5537.8  828.56  5607.9  829.87  5727.9  830.43
  5998.0  833.43  6148.1  836.62  6288.2  840.56  6508.3  840.49  6537.7  841.02
#Mann=3,-1,0
  4493.6    0.05       0  4994.5    0.04       0  5000.7    0.05       0
Bank Sta=4994.5,5000.7
Exp/Cntr=0.3,0.1

Type RM Length L Ch R = 1,7161,532,532,532
BEGIN DESCRIPTION:
MDW T 021 11.0
END DESCRIPTION:
XS GIS Cut Line= 3
      2288545.37      7108671.28      2287884.45      7108657.53
      2286354.41      7108653.92
#Sta/Elev= 30
  4354.8  839.16  4401.2  836.73  4431.2  832.89  4441.2  832.56  4531.2  833.49
  4541.2  832.12  4561.2  827.20  4571.2  826.09  4701.2  826.86  4731.2  822.19
  4741.2  821.69  4841.3  818.95  4871.3  817.39  4891.3  817.91  4981.3  816.26
  5001.3  814.10  5008.0  811.46  5009.0  810.96  5014.2  811.46  5021.3  811.49
  5031.3  814.99  5041.3  816.94  5051.3  817.28  5331.3  819.76  5551.3  825.39
  5651.3  825.71  5751.3  828.27  6181.3  835.16  6371.3  835.78  6545.9  839.34
#Mann=3,-1,0
  4354.8    0.05       0  5008.0    0.04       0  5014.2    0.05       0
Bank Sta=5008,5014.2
Exp/Cntr=0.3,0.1

Type RM Length L Ch R = 1,6629,384,384,384
BEGIN DESCRIPTION:
Mapping XS b0177e8c
END DESCRIPTION:
XS GIS Cut Line= 3
      2288211.93      7107992.13      2287602.17      7108550.92
      2287105.18      7108566.17
#Sta/Elev= 30
  4600.1  829.00  4607.6  828.50  4615.0  825.71  4621.8  825.21  4629.2  823.09
  4636.0  822.73  4643.4  820.83  4650.1  820.94  4657.5  819.62  4727.8  819.54
  4883.8  815.77  4961.5  815.42  4975.7  813.94  4989.9  810.23  5000.9  808.99
  5001.9  808.49  5007.3  808.99  5018.3  810.32  5025.1  812.00  5053.4  813.70
  5117.6  813.57  5166.9  814.54  5173.8  813.97  5216.2  814.83  5244.6  816.85
  5343.9  816.92  5520.4  819.29  5640.4  822.99  5700.5  823.03  5924.4  827.54
#Mann=3,-1,0
  4600.1    0.05       0  5000.9    0.04       0  5007.3    0.05       0
Bank Sta=5000.9,5007.3
Exp/Cntr=0.3,0.1

Type RM Length L Ch R = 1,6245,412,412,412
BEGIN DESCRIPTION:
MDW T 021 9.0
END DESCRIPTION:
XS GIS Cut Line= 3
      2288390.86      7107890.03      2287829.00      7107910.00
      2286599.18      7107961.21
#Sta/Elev= 30
  4434.1  846.28  4536.0  846.42  4577.5  844.20  4596.1  840.39  4626.1  831.61
  4646.1  828.91  4686.1  819.65  4696.1  818.73  4786.2  817.17  4826.2  814.30
  4956.3  811.60  4976.3  809.99  4986.3  807.76  5003.1  807.42  5004.2  806.92
  5009.5  807.42  5026.3  810.52  5056.4  811.59  5136.4  811.31  5166.5  810.27
  5196.5  811.34  5336.6  810.75  5346.6  809.94  5354.2  811.36  5359.2  810.67
  5376.6  819.80  5386.7  820.51  5566.8  824.11  5967.2  828.04  6227.2  833.95
#Mann=3,-1,0
  4434.1    0.05       0  5003.1    0.04       0  5009.5    0.05       0
Bank Sta=5003.1,5009.5
Exp/Cntr=0.3,0.1

Type RM Length L Ch R = 1,5833,518,518,518
BEGIN DESCRIPTION:
MDW T 021 8.0
END DESCRIPTION:
XS GIS Cut Line= 3
      2288573.16      7107525.45      2287778.94      7107514.97
      2286643.34      7107617.40
#Sta/Elev= 30
  4200.9  840.87  4245.1  841.57  4255.1  840.19  4265.1  841.23  4275.1  839.51
  4325.1  838.00  4395.1  831.59  4465.1  830.48  4485.1  831.18  4625.1  828.12
  4665.1  817.70  4725.1  811.68  4845.1  806.92  4915.1  807.12  4955.1  809.25
  4975.1  808.12  4985.1  806.57  4990.9  803.99  4991.9  803.49  4997.6  803.99
  5035.3  808.69  5135.7  809.47  5206.0  814.43  5346.5  818.76  5447.0  820.34
  5657.8  820.84  5878.7  825.87  5949.0  828.17  5995.8  831.09  6135.4  834.01
#Mann=3,-1,0
  4200.9    0.05       0  4990.9   0.033       0  4997.6    0.05       0
Bank Sta=4990.9,4997.6
Exp/Cntr=0.3,0.1

Type RM Length L Ch R = 1,5315,426,426,426
BEGIN DESCRIPTION:
MDW T 021 7.0
END DESCRIPTION:
XS GIS Cut Line= 3
      2288420.38      7107004.62      2287780.06      7107049.56
      2286673.06      7107165.97
#Sta/Elev= 30
  4358.1  832.69  4379.5  832.90  4399.6  831.11  4459.7  829.46  4469.8  828.13
  4550.0  826.75  4630.1  821.88  4640.2  820.78  4647.2  817.07  4670.2  810.11
  4700.3  803.76  4780.5  804.95  4830.6  803.58  4900.8  805.12  4920.9  804.15
  4950.9  804.80  4987.7  802.98  4988.7  802.48  4994.4  802.98  4998.0  804.23
  5011.1  804.81  5147.2  805.14  5192.1  807.02  5245.3  810.97  5322.8  809.89
  5431.4  810.95  5534.5  813.84  5634.5  818.42  5875.9  823.46  6113.1  831.03
#Mann=3,-1,0
  4358.1    0.05       0  4987.7    0.04       0  4994.4    0.05       0
Bank Sta=4987.7,4994.4
Exp/Cntr=0.3,0.1

Type RM Length L Ch R = 1,4889,249,249,249
BEGIN DESCRIPTION:
MDW T 021 6.0
END DESCRIPTION:
XS GIS Cut Line= 3
      2288390.87      7106521.30      2287879.36      7106649.59
      2287179.03      7106859.99
#Sta/Elev= 30
  4476.1  822.52  4601.7  821.08  4657.1  819.17  4693.1  815.00  4698.3  815.48
  4734.3  810.42  4780.6  810.76  4797.6  803.76  4816.6  802.10  4962.6  802.54
  4972.9  801.39  4977.9  799.38  4979.0  798.88  4984.8  799.38  4986.5  800.28
  5006.2  799.79  5020.9  802.47  5026.1  801.53  5059.1  802.91  5244.0  803.30
  5306.6  806.19  5390.2  804.40  5443.5  804.96  5504.3  807.24  5509.5  806.52
  5536.3  808.70  5542.6  811.10  5547.8  809.26  5575.6  814.65  5734.7  817.19
#Mann=3,-1,0
  4476.1    0.05       0  4977.9    0.04       0  4984.8    0.05       0
Bank Sta=4977.9,4984.8
Exp/Cntr=0.3,0.1

Type RM Length L Ch R = 1,4640,213,213,213
BEGIN DESCRIPTION:
MDW T 021 5.5
END DESCRIPTION:
XS GIS Cut Line= 3
      2288340.18      7106321.46      2287831.26      7106454.06
      2287128.95      7106742.65
#Sta/Elev= 30
  4478.5  814.75  4521.1  812.86  4541.7  812.80  4569.7  811.53  4574.9  811.94
  4610.2  809.92  4615.4  810.44  4650.7  808.04  4655.9  808.41  4767.0  802.65
  4913.7  800.37  4929.0  800.31  4944.7  801.89  4964.4  801.48  4969.5  798.36
  4982.6  798.04  4983.7  797.54  4989.5  798.04  5028.1  798.51  5039.3  802.01
  5050.1  802.14  5057.5  801.23  5086.9  801.61  5104.2  802.59  5110.8  804.38
  5116.2  803.97  5125.8  805.14  5179.8  807.61  5385.2  812.05  5763.7  816.97
#Mann=3,-1,0
  4478.5    0.05       0  4982.6   0.033       0  4989.5    0.05       0
Bank Sta=4982.6,4989.5
Exp/Cntr=0.3,0.1

Type RM Length L Ch R = 1,4427,598,598,598
BEGIN DESCRIPTION:
Mapping XS 9afe4cc8
END DESCRIPTION:
XS GIS Cut Line= 2
      2288287.09      7106314.44      2287413.51      7106200.33
#Sta/Elev= 30
  4536.7  811.95  4610.0  809.68  4615.5  808.61  4625.5  807.67  4645.7  806.83
  4696.1  803.69  4756.6  801.80  4776.8  800.67  4807.1  800.22  4836.7  800.31
  4867.6  799.55  4887.7  799.73  4920.7  800.69  4938.2  800.15  4988.6  799.85
  4994.6  798.45  4996.2  796.05  4997.3  795.55  5002.1  795.55  5003.1  796.05
  5008.8  797.07  5018.9  801.98  5028.9  802.72  5073.6  803.67  5079.4  804.15
  5109.6  805.09  5226.4  808.05  5231.4  807.89  5361.7  809.93  5417.7  810.28
#Mann=3,-1,0
  4536.7    0.05       0  4996.2   0.033       0  5003.1    0.05       0
Bank Sta=4996.2,5003.1
Exp/Cntr=0.3,0.1

Type RM Length L Ch R = 1,3829,304,304,304
BEGIN DESCRIPTION:
MDW T 021 5.0
END DESCRIPTION:
XS GIS Cut Line= 3
      2288571.75      7106207.58      2288179.01      7105868.08
      2287193.83      7105543.55
#Sta/Elev= 30
  4473.5  818.30  4615.5  813.51  4785.5  804.93  4913.3  801.09  4948.9  798.96
  4963.2  797.11  4969.8  797.93  4973.9  794.64  4975.0  794.14  4979.8  794.14
  4980.9  794.64  4984.1  795.25  4995.3  794.84  5000.2  796.50  5005.5  794.92
  5024.2  796.47  5032.0  797.97  5037.2  797.44  5045.3  799.23  5100.8  797.06
  5171.6  796.40  5286.2  799.63  5361.2  801.12  5424.3  803.35  5519.1  805.48
  5609.2  806.49  5729.7  805.63  5863.4  803.64  5908.6  802.25  6029.9  801.96
#Mann=3,-1,0
  4473.5    0.05       0  4973.9    0.04       0  4980.9    0.05       0
Bank Sta=4973.9,4980.9
Exp/Cntr=0.3,0.1

Type RM Length L Ch R = 1,3525,107,107,107
BEGIN DESCRIPTION:
MDW T 021 4.0
END DESCRIPTION:
XS GIS Cut Line= 4
      2288519.67      7106109.95      2288332.20      7105675.52
      2288018.35      7105211.48      2287244.63      7105367.70
#Sta/Elev= 30
  4528.2  815.05  4567.0  814.58  4572.4  813.75  4713.3  808.56  4794.9  804.32
  4865.5  801.94  4870.9  801.03  4917.9  799.45  4923.4  798.37  4941.4  798.14
  4946.9  797.28  4985.6  796.39  4993.9  793.38  5004.5  792.48  5005.6  791.98
  5011.5  792.48  5015.0  796.00  5021.1  796.24  5158.9  796.16  5201.2  796.93
  5317.6  796.02  5353.6  794.85  5374.6  796.91  5410.6  798.85  5628.5  802.98
  5815.9  803.89  5826.1  803.25  5933.2  803.82  6122.0  803.14  6350.9  800.14
#Mann=3,-1,0
  4528.2    0.05       0  5004.5    0.04       0  5011.5    0.05       0
Bank Sta=5004.5,5011.5
Exp/Cntr=0.3,0.1

Type RM Length L Ch R = 1,3418,436,436,436
BEGIN DESCRIPTION:
Mapping XS 109a4e1b
END DESCRIPTION:
XS GIS Cut Line= 2
      2288475.99      7105779.24      2288142.15      7104943.23
#Sta/Elev= 30
  4811.0  804.20  4875.2  801.23  4953.4  798.61  4971.7  796.81  4977.6  795.44
  4993.2  795.44  5001.9  793.49  5007.3  792.95  5014.8  795.17  5055.8  795.63
  5079.4  795.18  5100.9  796.32  5122.5  796.51  5294.7  794.69  5306.3  795.10
  5325.2  794.61  5337.8  795.25  5348.6  794.86  5356.7  791.46  5357.8  790.96
  5362.6  790.96  5363.7  791.46  5370.1  793.79  5379.1  794.89  5384.4  794.46
  5391.6  794.87  5414.1  796.99  5575.7  800.01  5629.6  800.59  5711.2  800.46
#Mann=3,-1,0
  4811.0    0.05       0  5356.7   0.033       0  5363.7    0.05       0
Bank Sta=5356.7,5363.7
Exp/Cntr=0.3,0.1

Type RM Length L Ch R = 1,2982,225,225,225
BEGIN DESCRIPTION:
Mapping XS ffa49520
END DESCRIPTION:
XS GIS Cut Line= 3
      2288691.09      7105638.46      2288539.54      7105317.59
      2288147.54      7104884.11
#Sta/Elev= 30
  4479.6  805.28  4489.0  804.26  4511.1  805.49  4523.6  803.92  4546.4  803.00
  4563.6  801.29  4591.9  801.66  4599.5  800.42  4665.9  798.21  4779.6  796.70
  4819.6  795.85  4825.1  795.02  4840.3  796.31  4854.5  794.92  4882.9  794.01
  4889.7  794.92  4925.5  793.90  4939.1  794.35  4953.2  793.30  4974.8  793.83
  4989.0  792.31  4995.8  789.72  4999.6  789.50  5000.7  789.00  5006.9  789.50
  5017.4  790.91  5024.2  793.60  5060.0  793.53  5279.0  799.11  5418.9  800.28
#Mann=3,-1,0
  4479.6    0.05       0  4999.6    0.04       0  5006.9    0.05       0
Bank Sta=4999.6,5006.9
Exp/Cntr=0.3,0.1

Type RM Length L Ch R = 1,2757,363,363,363
BEGIN DESCRIPTION:
Mapping XS 51e0cc9a
END DESCRIPTION:
XS GIS Cut Line= 2
      2288918.44      7105292.07      2288192.99      7104729.38
#Sta/Elev= 30
  4571.8  798.95  4594.9  798.61  4615.7  797.28  4622.0  797.88  4679.9  797.15
  4708.9  796.23  4758.7  795.54  4829.3  793.43  4858.3  793.92  4872.8  793.03
  4887.2  793.43  4922.5  792.92  4986.8  793.44  4993.1  791.90  4997.7  789.89
  4998.8  789.39  5003.8  789.39  5005.0  789.89  5007.6  791.72  5022.1  793.46
  5036.6  793.41  5042.9  792.66  5092.7  791.37  5121.7  792.86  5157.0  793.36
  5178.6  794.46  5250.2  796.20  5320.8  796.99  5393.3  798.55  5489.9  798.87
#Mann=3,-1,0
  4571.8    0.05       0  4997.7   0.033       0  5005.0    0.05       0
Bank Sta=4997.7,5005
Exp/Cntr=0.3,0.1

Type RM Length L Ch R = 1,2394,390,390,390
BEGIN DESCRIPTION:
MDW T 021 3.0
END DESCRIPTION:
XS GIS Cut Line= 3
      2289403.96      7104930.49      2288629.40      7104694.84
      2288050.02      7104624.96
#Sta/Elev= 30
  4189.4  801.62  4247.4  799.77  4476.8  796.89  4497.7  795.81  4508.2  796.88
  4520.7  797.11  4529.1  796.71  4539.5  795.28  4548.3  795.99  4624.5  795.17
  4696.3  793.51  4706.8  794.21  4723.0  792.82  4826.8  791.07  4849.4  789.70
  4850.6  789.20  4855.7  789.20  4856.8  789.70  4874.0  790.38  4957.6  791.16
  5009.5  790.00  5029.6  792.08  5130.4  792.05  5165.2  791.47  5180.7  793.08
  5200.9  793.77  5372.1  798.23  5503.4  798.48  5523.2  799.15  5582.6  798.27
#Mann=3,-1,0
  4189.4    0.05       0  4849.4   0.033       0  4856.8    0.05       0
Bank Sta=4849.4,4856.8
Exp/Cntr=0.3,0.1

Type RM Length L Ch R = 1,2004,444,444,444
BEGIN DESCRIPTION:
MDW T 021 2.0
END DESCRIPTION:
XS GIS Cut Line= 3
      2289436.45      7104747.52      2288646.13      7104343.52
      2288152.83      7104315.27
#Sta/Elev= 30
  4084.4  795.74  4349.5  793.41  4421.8  791.58  4438.4  793.38  4452.2  793.29
  4466.2  791.43  4527.3  791.59  4643.9  790.09  4721.6  789.76  4766.0  790.81
  4771.6  790.15  4777.8  790.97  4800.3  789.97  4810.4  790.49  4838.3  789.45
  4854.9  790.00  4899.3  788.83  4921.5  789.99  4949.4  790.29  4957.5  788.00
  4985.5  787.47  4986.6  786.97  4992.9  787.47  5019.2  790.79  5109.3  794.25
  5149.4  795.06  5219.5  795.99  5229.5  795.38  5419.9  795.96  5466.1  796.81
#Mann=3,-1,0
  4084.4    0.05       0  4985.5   0.033       0  4992.9    0.05       0
Bank Sta=4985.5,4992.9
Exp/Cntr=0.3,0.1

Type RM Length L Ch R = 1,1560,427,427,427
BEGIN DESCRIPTION:
Mapping XS 99a1bc27
END DESCRIPTION:
XS GIS Cut Line= 3
      2289370.47      7104572.47      2289058.29      7103958.35
      2288372.86      7103886.49
#Sta/Elev= 30
  3972.4  792.10  4095.0  790.34  4139.5  790.64  4189.6  789.52  4367.8  788.75
  4400.9  787.93  4428.8  789.23  4457.5  789.05  4489.9  787.46  4534.4  788.60
  4584.5  787.91  4637.0  788.08  4670.7  788.96  4689.6  788.42  4710.9  788.82
  4761.1  787.21  4787.8  788.58  4811.4  788.90  4932.1  788.16  4979.2  788.54
  4984.3  788.35  4988.7  785.17  4989.9  784.67  4996.1  785.17  5002.5  785.67
  5012.5  788.64  5032.6  789.76  5093.0  790.09  5170.7  792.03  5350.5  793.00
#Mann=3,-1,0
  3972.4    0.05       0  4988.7   0.033       0  4996.1    0.05       0
Bank Sta=4988.7,4996.1
Exp/Cntr=0.3,0.1

Type RM Length L Ch R = 1,1133,0,0,0
BEGIN DESCRIPTION:
MDW T 021 1.0
END DESCRIPTION:
XS GIS Cut Line= 3
      2289453.34      7104455.84      2288778.52      7103504.80
      2288086.16      7104121.62
#Sta/Elev= 30
  3842.0  790.28  4229.3  787.38  4236.9  788.53  4278.7  789.15  4287.3  787.62
  4308.2  788.94  4388.2  788.96  4394.3  787.81  4400.9  788.96  4430.0  788.39
  4437.7  789.37  4480.4  788.04  4523.5  788.56  4572.7  786.40  4652.7  787.90
  4709.2  785.43  4768.3  787.38  4982.4  786.43  4997.1  784.54  4999.5  782.54
  5000.7  782.04  5007.0  782.54  5008.0  783.39  5011.3  782.54  5018.8  786.53
  5033.0  786.82  5089.1  786.67  5380.0  791.62  5797.7  796.35  5935.4  796.35
#Mann=3,-1,0
  3842.0    0.05       0  4999.5   0.033       0  5007.0    0.05       0
Bank Sta=4999.5,5007
Exp/Cntr=0.3,0.1
