--- MDW T 049.prj (project) ---

Proj Title=MDW T 049 Base Level Engineering
Current Plan=p01
Default Exp/Contr=0.3,0.1
English Units
Geom File=g01
Flow File=f01
Plan File=p01
BEGIN DESCRIPTION:
MDW T 049
END DESCRIPTION:

--- MDW T 049.p01 (plan) ---

Plan Title=Multiple Run
Short Identifier=Multiple
Geom File=g01
Flow File=f01
Subcritical Flow
K Sum by GR= 0
Std Step Tol= 0.01
Critical Tol= 0.01
Num of Std Step Trials= 20
Max Error Tol= 0.3
Flow Tol Ratio= 0.001
Split Flow NTrial= 30
Split Flow Tol= 0.02
Split Flow Ratio= 0.02
Log Output Level= 0
Friction Slope Method= 1
Unsteady Friction Slope Method= 2
Unsteady Bridges Friction Slope Method= 1
Parabolic Critical Depth
Global Vel Dist=  1 , 1 , 1
Global Log Level= 0
CheckData=True
Encroach Param= -1, 0, 0, 0
BEGIN DESCRIPTION:
Multiple Run
END DESCRIPTION:

--- MDW T 049.f01 (steady flow) ---

Flow Title=Multiple
Number of Profiles=7
Profile Names=10-year,25-year,50-year,1pct_min,100-year,1pct_plu,500-year
River Rch & RM= MDW T 049,Reach-1,18556
     555     754     917     554    1105    2204    1607
River Rch & RM= MDW T 049,Reach-1,15320
     940    1320    1641    1012    2019    4028    3063
River Rch & RM= MDW T 049,Reach-1,6124
    1131    1605    2010    1247    2489    4966    3827
Boundary for River Rch & Prof#=MDW T 049,Reach-1,1
Up Type=0
Dn Type=3
Dn Slope=0.005
Boundary for River Rch & Prof#=MDW T 049,Reach-1,2
Up Type=0
Dn Type=3
Dn Slope=0.005
Boundary for River Rch & Prof#=MDW T 049,Reach-1,3
Up Type=0
Dn Type=3
Dn Slope=0.005
Boundary for River Rch & Prof#=MDW T 049,Reach-1,4
Up Type=0
Dn Type=3
Dn Slope=0.005
Boundary for River Rch & Prof#=MDW T 049,Reach-1,5
Up Type=0
Dn Type=3
Dn Slope=0.005
Boundary for River Rch & Prof#=MDW T 049,Reach-1,6
Up Type=0
Dn Type=3
Dn Slope=0.005
Boundary for River Rch & Prof#=MDW T 049,Reach-1,7
Up Type=0
Dn Type=3
Dn Slope=0.005

--- MDW T 049.g01 (geometry) ---

Geom Title=Existing Conditions

River Reach=MDW T 049,Reach-1
Reach XY= 30
      2299429.00      7086710.00      2300265.55      7087039.02
      2300500.39      7087450.97      2301612.78      7088076.15
      2302155.93      7087998.15      2302418.58      7088420.24
      2302879.94      7088443.48      2303184.78      7088888.15
      2303620.82      7088813.43      2303713.66      7089185.13
      2303975.55      7089311.25      2304030.22      7089956.57
      2304744.86      7089744.39      2304946.74      7089935.89
      2305523.29      7089532.40      2306128.60      7090137.67
      2306882.76      7089872.58      2307699.54      7089859.47
      2308015.36      7089936.16      2308056.53      7090251.43
      2308561.47      7090360.07      2308479.89      7090849.41
      2308884.35      7091632.66      2308798.00      7092458.18
      2308948.26      7092634.41      2308663.11      7092785.12
      2308850.23      7093292.55      2308653.94      7093359.34
      2308376.30      7093975.01      2308879.00      7094310.00

Type RM Length L Ch R = 1,18556,328,328,328
BEGIN DESCRIPTION:
MDW T 049 40.0
END DESCRIPTION:
XS GIS Cut Line= 3
      2299402.50      7086956.00      2299529.00      7086810.00
      2299779.85      7086283.82
#Sta/Elev= 30
  4822.3  878.59  4873.5  877.54  4909.6  876.04  4930.5  876.06  4944.7  875.72
  4987.5  872.38  4992.1  871.69  4992.4  871.19  4995.9  871.19  4996.1  871.69
  5001.7  872.17  5082.0  874.02  5159.5  875.15  5194.0  876.39  5256.6  877.04
  5270.3  876.78  5279.3  877.28  5324.7  877.95  5336.8  878.57  5347.4  878.45
  5352.9  878.96  5358.9  878.70  5375.6  879.40  5381.1  878.87  5392.1  878.89
  5398.3  879.30  5403.8  878.64  5421.0  879.10  5426.5  878.75  5598.4  880.90
#Mann=3,-1,0
  4822.3    0.05       0  4992.1   0.033       0  4996.1    0.05       0
Bank Sta=4992.1,4996.1
Exp/Cntr=0.3,0.1

Type RM Length L Ch R = 1,18228,374,374,374
BEGIN DESCRIPTION:
MDW T 049 39.0
END DESCRIPTION:
XS GIS Cut Line= 3
      2299402.80      7087474.04      2299818.81      7086909.55
      2300073.40      7086341.19
#Sta/Elev= 30
  4301.9  883.19  4331.6  882.86  4337.8  881.57  4373.3  879.50  4780.5  875.00
  4803.6  875.42  4816.2  874.84  4824.4  872.53  4845.3  870.25  4853.5  871.19
  4859.9  873.21  4874.6  873.77  4895.4  872.86  4910.1  873.31  4966.4  872.05
  4981.0  872.75  4989.5  871.41  4995.7  871.43  4997.7  869.88  4998.0  869.38
  5001.5  869.38  5001.7  869.88  5005.6  869.88  5012.0  872.51  5017.4  871.86
  5024.5  872.46  5069.3  871.67  5123.2  872.93  5358.5  875.41  5625.9  880.64
#Mann=3,-1,0
  4301.9    0.05       0  4997.7   0.033       0  5001.7    0.05       0
Bank Sta=4997.7,5001.7
Exp/Cntr=0.3,0.1

Type RM Length L Ch R = 1,17854,446,446,446
BEGIN DESCRIPTION:
MDW T 049 38.0
END DESCRIPTION:
XS GIS Cut Line= 3
      2299674.10      7087500.03      2300158.87      7087010.31
      2300592.04      7086336.87
#Sta/Elev= 30
  4309.3  875.95  4425.9  873.94  4510.8  873.15  4588.6  873.62  4800.7  871.78
  4878.5  870.00  4892.6  869.27  4899.7  868.04  4906.8  867.77  4913.9  869.40
  4928.0  869.73  4977.5  869.27  4991.6  867.22  4993.1  865.19  4993.3  864.69
  4996.8  864.69  4997.1  865.19  5001.5  865.19  5006.3  868.34  5070.1  871.27
  5165.2  872.47  5302.8  875.82  5354.3  875.96  5403.0  877.88  5700.3  883.11
  5729.4  884.09  5744.6  883.94  5750.5  884.68  5771.6  885.57  5799.1  885.82
#Mann=3,-1,0
  4309.3    0.05       0  4993.1   0.033       0  4997.1    0.05       0
Bank Sta=4993.1,4997.1
Exp/Cntr=0.3,0.1

Type RM Length L Ch R = 1,17408,177,177,177
BEGIN DESCRIPTION:
MDW T 049 37.0
END DESCRIPTION:
XS GIS Cut Line= 3
      2299778.99      7087860.00      2300408.69      7087340.14
      2300734.66      7086780.63
#Sta/Elev= 30
  4182.2  878.78  4374.4  874.43  4402.7  875.82  4416.0  875.50  4423.9  873.46
  4459.0  873.75  4502.1  872.48  4508.5  870.43  4516.4  870.29  4522.9  872.53
  4530.7  872.30  4537.2  873.30  4565.9  872.70  4572.4  871.02  4586.7  870.52
  4885.1  867.44  4977.6  865.51  4993.7  863.17  4994.0  862.67  4997.7  863.17
  5007.0  863.25  5028.5  865.51  5034.3  867.75  5241.9  871.08  5392.5  875.60
  5429.7  878.12  5584.4  879.29  5627.4  881.36  5643.1  887.17  5646.3  887.43
#Mann=3,-1,0
  4182.2    0.05       0  4993.7   0.033       0  4997.7    0.05       0
Bank Sta=4993.7,4997.7
Exp/Cntr=0.3,0.1

Type RM Length L Ch R = 1,17231,233,233,233
BEGIN DESCRIPTION:
Mapping XS 179dbb92
END DESCRIPTION:
XS GIS Cut Line= 3
      2300259.82      7087531.23      2300472.71      7087550.74
      2300667.20      7087236.78
#Sta/Elev= 30
  4689.4  868.57  4718.7  868.20  4748.8  868.22  4809.1  866.40  4819.1  865.71
  4849.2  865.12  4879.4  865.09  4907.8  864.23  4923.2  864.59  4944.4  863.84
  4959.8  863.99  4965.7  863.50  4974.6  863.51  4981.1  863.12  5000.3  859.90
  5000.6  859.40  5004.1  859.40  5004.3  859.90  5009.9  860.44  5033.1  865.67
  5054.3  866.72  5060.2  866.61  5170.1  868.91  5176.0  868.67  5185.5  868.95
  5191.4  868.72  5243.4  869.15  5249.3  869.33  5264.6  870.59  5272.5  870.31
#Mann=3,-1,0
  4689.4    0.05       0  5000.3   0.033       0  5004.3    0.05       0
Bank Sta=5000.3,5004.3
Exp/Cntr=0.3,0.1

Type RM Length L Ch R = 1,16998,172,172,172
BEGIN DESCRIPTION:
Mapping XS 3c0938c9
END DESCRIPTION:
XS GIS Cut Line= 4
      2300235.29      7087571.58      2300605.30      7087583.36
      2300760.91      7087598.90      2300880.53      7087334.25
#Sta/Elev= 30
  4515.0  869.00  4548.7  867.89  4628.8  866.90  4678.8  865.56  4758.8  864.14
  4838.9  863.69  4897.8  862.33  4909.0  862.84  4959.3  861.54  4989.4  859.79
  4998.4  860.41  5001.4  859.72  5001.7  859.22  5005.2  859.22  5005.4  859.72
  5019.6  860.34  5043.7  860.24  5047.5  860.80  5070.6  861.73  5099.2  862.27
  5106.2  862.86  5122.3  862.98  5145.4  863.97  5150.9  863.70  5214.7  865.06
  5243.3  864.73  5259.9  865.11  5303.7  866.93  5318.2  867.16  5332.0  868.03
#Mann=3,-1,0
  4515.0    0.05       0  5001.4   0.033       0  5005.4    0.05       0
Bank Sta=5001.4,5005.4
Exp/Cntr=0.3,0.1

Type RM Length L Ch R = 1,16826,177,177,177
BEGIN DESCRIPTION:
Mapping XS 2d16469f
END DESCRIPTION:
XS GIS Cut Line= 4
      2300521.79      7087885.00      2300681.35      7087679.67
      2301160.08      7087708.50      2301184.53      7087642.63
#Sta/Elev= 30
  4568.0  866.68  4762.6  863.33  4768.9  863.84  4783.4  863.45  4789.7  862.93
  4797.9  862.97  4804.2  862.48  4935.9  861.65  4945.9  861.32  4955.9  860.15
  4965.9  859.53  4996.0  858.37  5014.0  857.08  5014.3  856.58  5017.8  856.58
  5018.0  857.08  5026.0  857.40  5036.1  858.42  5066.1  858.34  5082.1  859.44
  5087.1  857.96  5126.2  859.63  5196.4  858.66  5216.4  858.82  5256.5  858.06
  5307.6  857.78  5338.0  859.08  5345.5  860.01  5350.8  859.96  5377.9  862.43
#Mann=3,-1,0
  4568.0    0.05       0  5014.0   0.033       0  5018.0    0.05       0
Bank Sta=5014,5018
Exp/Cntr=0.3,0.1

Type RM Length L Ch R = 1,16649,149,149,149
BEGIN DESCRIPTION:
Mapping XS 24aee1d6
END DESCRIPTION:
XS GIS Cut Line= 4
      2300878.64      7087927.23      2301046.53      7087723.32
      2301173.98      7087728.97      2301202.03      7087641.04
#Sta/Elev= 30
  4786.8  863.25  4806.8  863.02  4813.3  862.64  4821.1  862.71  4827.6  862.29
  4856.3  862.39  4862.8  862.04  4877.1  861.87  4912.7  860.80  4948.8  860.76
  4969.7  860.46  4977.5  859.62  4984.0  858.27  4990.5  857.69  4998.3  856.32
  5002.8  856.19  5003.1  855.69  5006.6  855.69  5006.8  856.19  5027.0  857.47
  5041.4  859.10  5143.5  858.25  5173.5  857.56  5187.9  857.56  5207.6  858.27
  5212.8  858.19  5239.8  859.96  5245.0  859.88  5268.7  862.49  5270.8  862.49
#Mann=3,-1,0
  4786.8    0.05       0  5002.8   0.033       0  5006.8    0.05       0
Bank Sta=5002.8,5006.8
Exp/Cntr=0.3,0.1

Type RM Length L Ch R = 1,16500,157,157,157
BEGIN DESCRIPTION:
Mapping XS c56ecdcc
END DESCRIPTION:
XS GIS Cut Line= 2
      2301016.36      7088162.79      2301220.27      7087640.91
#Sta/Elev= 30
  4638.4  861.62  4712.8  861.26  4718.1  860.98  4767.1  860.65  4802.4  859.75
  4821.4  860.10  4826.8  859.93  4845.4  860.81  4851.2  859.73  4875.7  859.74
  4905.6  859.05  4930.0  857.72  4952.7  857.54  4959.9  856.84  4963.3  856.19
  4963.5  855.69  4967.0  855.69  4967.3  856.19  5027.9  856.39  5044.0  858.02
  5060.1  857.78  5068.5  858.11  5103.7  857.43  5146.0  858.44  5152.7  859.03
  5158.1  859.05  5177.2  860.69  5182.5  860.64  5196.5  862.52  5198.7  862.52
#Mann=3,-1,0
  4638.4    0.05       0  4963.3   0.033       0  4967.3    0.05       0
Bank Sta=4963.3,4967.3
Exp/Cntr=0.3,0.1

Type RM Length L Ch R = 1,16343,114,114,114
BEGIN DESCRIPTION:
Mapping XS 25519c4c
END DESCRIPTION:
XS GIS Cut Line= 2
      2301293.20      7088279.05      2301296.72      7087640.46
#Sta/Elev= 30
  4597.8  858.77  4646.9  858.70  4742.5  858.16  4816.9  856.90  4846.9  856.89
  4876.9  856.35  4886.9  856.47  4896.9  858.10  4906.9  858.83  4936.9  858.45
  4956.9  857.34  4966.9  856.52  4976.9  856.28  4996.9  856.40  5004.9  856.24
  5005.1  855.74  5008.6  855.74  5008.9  856.24  5016.9  856.45  5046.9  856.35
  5056.9  856.82  5116.9  857.33  5146.9  857.96  5156.9  858.58  5196.9  859.48
  5206.9  859.93  5216.9  860.77  5226.9  862.45  5234.1  863.27  5236.4  863.27
#Mann=3,-1,0
  4597.8    0.05       0  5004.9   0.033       0  5008.9    0.05       0
Bank Sta=5004.9,5008.9
Exp/Cntr=0.3,0.1

Type RM Length L Ch R = 1,16229,305,305,305
BEGIN DESCRIPTION:
Mapping XS e7443886
END DESCRIPTION:
XS GIS Cut Line= 2
      2301400.24      7088294.12      2301404.88      7087684.04
#Sta/Elev= 30
  4620.6  857.71  4644.7  857.73  4664.7  857.53  4694.7  857.40  4754.7  856.65
  4794.7  855.94  4814.7  855.39  4834.7  855.24  4844.7  855.40  4854.7  855.27
  4864.7  854.93  4874.7  854.84  4904.7  854.97  4954.7  855.93  4964.7  855.93
  4974.7  855.37  4992.7  853.47  4993.0  852.97  4996.5  852.97  4996.7  853.47
  5004.7  853.70  5014.7  853.69  5034.7  854.79  5054.7  856.16  5074.7  857.34
  5084.7  857.24  5094.7  857.56  5112.5  857.71  5154.7  858.97  5230.7  860.56
#Mann=3,-1,0
  4620.6    0.05       0  4992.7   0.033       0  4996.7    0.05       0
Bank Sta=4992.7,4996.7
Exp/Cntr=0.3,0.1

Type RM Length L Ch R = 1,15924,193,193,193
BEGIN DESCRIPTION:
Mapping XS 3aaf9ba2
END DESCRIPTION:
XS GIS Cut Line= 2
      2301568.23      7088356.35      2301744.01      7087737.11
#Sta/Elev= 30
  4723.3  855.80  4761.1  855.67  4778.9  855.43  4784.1  854.95  4844.2  854.53
  4885.8  853.85  4924.9  852.10  4948.2  852.69  4979.4  853.05  4989.8  852.27
  4995.9  850.69  4996.1  850.19  4999.6  850.19  4999.9  850.69  5003.1  851.88
  5010.6  853.01  5031.4  853.28  5042.2  852.70  5083.3  852.06  5093.7  852.21
  5110.0  852.86  5183.0  854.41  5188.2  854.23  5239.3  854.48  5249.7  854.73
  5289.9  856.70  5329.0  857.88  5334.2  857.68  5362.9  858.43  5367.0  858.19
#Mann=3,-1,0
  4723.3    0.05       0  4995.9   0.033       0  4999.9    0.05       0
Bank Sta=4995.9,4999.9
Exp/Cntr=0.3,0.1

Type RM Length L Ch R = 1,15731,411,411,411
BEGIN DESCRIPTION:
Mapping XS e3a3f742
END DESCRIPTION:
XS GIS Cut Line= 3
      2301612.42      7088545.35      2301825.58      7088364.09
      2301838.03      7087807.24
#Sta/Elev= 30
  4476.0  856.56  4484.6  856.54  4505.9  855.73  4512.4  855.67  4520.1  855.11
  4583.8  854.51  4604.7  854.56  4612.4  854.36  4619.0  854.50  4676.1  853.88
  4696.9  853.85  4747.2  853.18  4809.9  852.73  4899.9  852.39  4919.9  852.18
  4949.9  851.55  4980.0  851.74  4990.0  851.48  4998.0  849.18  4998.2  848.68
  5001.7  848.68  5002.0  849.18  5010.0  851.77  5020.0  851.41  5030.0  851.36
  5070.0  851.74  5133.8  852.00  5170.0  852.42  5220.0  853.50  5312.8  856.14
#Mann=3,-1,0
  4476.0    0.05       0  4998.0   0.033       0  5002.0    0.05       0
Bank Sta=4998,5002
Exp/Cntr=0.3,0.1

Type RM Length L Ch R = 1,15320,47,47,47
BEGIN DESCRIPTION:
Mapping XS 41b6b503
END DESCRIPTION:
XS GIS Cut Line= 4
      2301922.63      7088325.44      2301945.81      7088188.46
      2302127.79      7088065.10      2302322.96      7087874.03
#Sta/Elev= 30
  4580.4  852.87  4589.8  852.29  4697.5  851.56  4742.3  850.85  4799.2  850.42
  4814.2  850.01  4844.0  849.94  4850.1  849.65  4865.1  849.62  4878.0  848.96
  4878.3  848.46  4881.8  848.46  4882.0  848.96  4886.1  849.22  4892.3  850.39
  4901.0  850.90  4907.1  851.67  4939.2  851.50  4943.6  851.78  4960.1  851.89
  5035.6  851.34  5056.7  851.70  5063.9  852.46  5085.0  853.28  5092.2  853.92
  5120.5  854.69  5141.6  854.42  5161.1  855.19  5198.2  856.41  5212.3  857.16
#Mann=5,-1,0
  4580.4    0.05       0  4878.0    0.07       0  4882.0    0.05       0
  4960.1    0.12       0  5161.1    0.05       0
Bank Sta=4878,4882
Exp/Cntr=0.3,0.1

Type RM Length L Ch R = 1,15273,135,135,135
BEGIN DESCRIPTION:
Mapping XS 61191769
END DESCRIPTION:
XS GIS Cut Line= 2
      2301936.69      7088308.22      2302350.58      7087916.46
#Sta/Elev= 30
  4642.5  851.87  4649.9  852.10  4671.3  851.85  4685.5  851.28  4720.7  850.87
  4777.3  849.43  4848.1  848.90  4869.1  849.03  4897.4  848.48  4918.9  848.68
  4933.0  847.63  4947.2  847.29  4954.1  847.62  4982.4  847.16  4989.7  846.62
  4996.6  846.56  5001.7  845.89  5001.9  845.39  5005.4  845.39  5005.7  845.89
  5010.7  847.06  5017.6  847.30  5024.9  848.67  5034.4  849.72  5045.9  851.58
  5060.1  852.57  5124.0  854.07  5145.0  855.18  5154.4  855.34  5212.4  856.25
#Mann=5,-1,0
  4642.5    0.05       0  5001.7   0.033       0  5005.7    0.05       0
  5034.4    0.12       0  5154.4    0.05       0
Bank Sta=5001.7,5005.7
Exp/Cntr=0.3,0.1

Type RM Length L Ch R = 1,15138,385,385,385
BEGIN DESCRIPTION:
Mapping XS 974b52f9
END DESCRIPTION:
XS GIS Cut Line= 3
      2301932.15      7088508.24      2302043.22      7088395.93
      2302449.84      7087984.80
#Sta/Elev= 30
  4547.0  853.02  4550.6  852.55  4614.3  851.93  4769.8  849.00  4812.2  848.53
  4833.5  848.90  4854.6  847.99  4882.9  847.85  4897.1  847.09  4925.3  847.57
  4939.5  847.27  4946.6  847.63  4960.7  847.54  5001.2  845.73  5001.4  845.23
  5004.9  845.23  5005.2  845.73  5017.3  846.71  5052.6  846.84  5102.2  850.63
  5116.3  851.32  5130.4  851.37  5144.6  852.20  5172.9  852.98  5179.9  852.70
  5187.0  853.22  5222.3  853.80  5257.7  855.56  5278.9  856.33  5283.2  856.05
#Mann=3,-1,0
  4547.0    0.05       0  5001.2   0.033       0  5005.2    0.05       0
Bank Sta=5001.2,5005.2
Exp/Cntr=0.3,0.1

Type RM Length L Ch R = 1,14753,269,269,269
BEGIN DESCRIPTION:
Mapping XS 466ffe3d
END DESCRIPTION:
XS GIS Cut Line= 3
      2302452.81      7088767.79      2302463.56      7088612.40
      2302502.12      7088054.69
#Sta/Elev= 30
  4668.5  847.73  4756.5  847.29  4816.6  846.41  4876.8  846.52  4946.9  845.39
  4967.0  845.46  4978.9  844.80  4987.0  843.59  4997.1  841.37  5004.9  840.50
  5005.3  840.00  5008.9  840.00  5009.3  840.50  5017.1  842.20  5027.1  842.98
  5047.2  843.18  5057.2  842.93  5077.3  843.84  5121.5  844.53  5147.4  845.91
  5197.5  847.57  5217.6  848.55  5237.6  849.96  5257.7  850.53  5264.2  851.08
  5287.8  851.38  5307.8  852.50  5347.9  853.51  5378.0  854.69  5383.3  855.33
#Mann=3,-1,0
  4668.5    0.05       0  5004.9   0.033       0  5009.3    0.05       0
Bank Sta=5004.9,5009.3
Exp/Cntr=0.3,0.1

Type RM Length L Ch R = 1,14484,350,350,350
BEGIN DESCRIPTION:
Mapping XS 0e89e2b0
END DESCRIPTION:
XS GIS Cut Line= 3
      2302674.48      7088785.43      2302697.33      7088639.50
      2302765.34      7088205.00
#Sta/Elev= 30
  4613.2  845.04  4628.8  844.36  4649.1  844.04  4669.3  844.06  4679.6  843.73
  4730.0  843.24  4750.3  842.77  4872.8  841.68  4922.3  841.59  4935.5  838.35
  4942.6  836.21  4950.5  835.98  4950.9  835.48  4954.5  835.48  4954.9  835.98
  4962.8  837.61  4973.0  838.88  4983.1  840.95  4993.1  838.58  4998.1  838.00
  5013.4  839.01  5023.6  837.90  5043.8  843.10  5065.9  843.70  5084.3  844.84
  5123.5  846.73  5128.6  846.51  5191.3  849.95  5196.4  849.98  5200.7  850.87
#Mann=3,-1,0
  4613.2    0.05       0  4950.5   0.033       0  4954.9    0.05       0
#XS Ineff=1,-1
 4982.20 5131.70  844.87
Permanent Ineff=
       F
Bank Sta=4950.5,4954.9
Exp/Cntr=0.3,0.1

Type RM Length L Ch R = 1,14134,182,182,182
BEGIN DESCRIPTION:
Mapping XS 7745579c
END DESCRIPTION:
XS GIS Cut Line= 2
      2302760.65      7088767.01      2303054.95      7088493.02
#Sta/Elev= 30
  4806.1  843.29  4824.0  842.79  4866.5  840.91  4873.4  840.76  4901.7  838.99
  4909.0  838.17  4944.2  837.09  4951.6  836.65  4965.7  836.38  4979.9  835.73
  4984.5  834.78  4984.9  834.28  4988.5  834.28  4988.9  834.78  4994.1  835.62
  5000.9  836.15  5008.2  836.08  5029.2  836.36  5043.4  836.08  5050.2  836.24
  5071.7  835.89  5085.9  835.97  5092.7  836.29  5106.9  838.17  5121.1  838.99
  5142.6  839.57  5149.4  840.12  5185.1  841.43  5191.9  841.88  5208.2  842.52
#Mann=3,-1,0
  4806.1    0.05       0  4984.5   0.033       0  4988.9    0.05       0
Bank Sta=4984.5,4988.9
Exp/Cntr=0.3,0.1

Type RM Length L Ch R = 1,13952,219,219,219
BEGIN DESCRIPTION:
Mapping XS 316f4e21
END DESCRIPTION:
XS GIS Cut Line= 2
      2302917.88      7088887.68      2303167.23      7088556.94
#Sta/Elev= 30
  4748.7  839.48  4755.5  839.69  4776.3  839.05  4790.9  839.29  4797.1  838.99
  4805.4  839.10  4811.7  838.32  4820.0  838.13  4826.3  837.01  4847.1  835.17
  4861.7  834.23  4883.6  833.83  4905.4  833.92  4911.6  833.62  4940.8  834.56
  4955.3  834.57  4990.7  833.46  4994.8  832.34  4995.2  831.84  4998.8  831.84
  4999.2  832.34  5005.3  832.52  5011.5  835.06  5019.8  836.14  5040.7  837.13
  5076.1  837.88  5090.6  838.84  5146.9  840.50  5155.2  841.12  5162.9  841.14
#Mann=3,-1,0
  4748.7    0.05       0  4994.8   0.033       0  4999.2    0.05       0
Bank Sta=4994.8,4999.2
Exp/Cntr=0.3,0.1

Type RM Length L Ch R = 1,13733,180,180,180
BEGIN DESCRIPTION:
Mapping XS b730cb58
END DESCRIPTION:
XS GIS Cut Line= 2
      2303117.27      7089041.32      2303214.22      7088571.52
#Sta/Elev= 30
  4819.5  838.01  4882.1  835.65  4892.3  835.70  4899.9  836.23  4905.0  835.95
  4912.7  836.25  4933.2  834.65  4950.1  832.97  4955.2  832.92  4984.2  831.25
  4992.1  828.26  4992.6  827.76  4996.2  827.76  4996.7  828.26  5000.4  830.66
  5014.9  832.17  5050.7  832.26  5055.8  831.84  5065.9  831.82  5117.0  832.00
  5146.1  833.10  5151.2  832.96  5157.8  833.64  5196.4  835.86  5201.5  835.73
  5239.5  837.73  5246.6  838.37  5290.5  839.93  5296.9  840.64  5299.2  840.55
#Mann=3,-1,0
  4819.5    0.05       0  4992.1   0.033       0  4996.7    0.05       0
Bank Sta=4992.1,4996.7
Exp/Cntr=0.3,0.1

Type RM Length L Ch R = 1,13553,298,298,298
BEGIN DESCRIPTION:
Mapping XS e33e2b74
END DESCRIPTION:
XS GIS Cut Line= 2
      2303324.27      7089043.41      2303297.86      7088605.91
#Sta/Elev= 30
  4857.3  834.61  4863.8  834.38  4880.8  834.83  4900.8  833.17  4920.8  832.36
  4950.9  832.01  4960.9  831.71  4970.9  832.02  4980.9  832.01  4991.0  828.75
  4998.7  828.43  4999.2  827.93  5002.8  827.93  5003.3  828.43  5011.0  830.00
  5026.9  829.96  5031.9  830.37  5051.1  830.43  5071.1  830.10  5081.1  830.16
  5111.2  829.49  5121.2  829.49  5151.2  830.19  5181.3  831.48  5195.0  832.25
  5201.3  832.95  5221.4  834.32  5271.5  836.97  5281.5  837.66  5295.6  837.72
#Mann=3,-1,0
  4857.3    0.05       0  4998.7   0.033       0  5003.3    0.05       0
Bank Sta=4998.7,5003.3
Exp/Cntr=0.3,0.1

Type RM Length L Ch R = 1,13255,211,211,211
BEGIN DESCRIPTION:
Mapping XS 9e235e00
END DESCRIPTION:
XS GIS Cut Line= 3
      2303349.64      7089052.34      2303474.24      7088984.36
      2303548.99      7088628.05
#Sta/Elev= 30
  4630.5  834.78  4640.6  834.97  4733.7  831.12  4765.9  831.24  4771.6  830.20
  4807.5  828.79  4821.4  830.24  4828.0  834.21  4838.2  835.00  4858.6  834.67
  4889.3  833.07  4916.1  830.94  4960.8  828.64  4966.0  827.63  4971.1  827.92
  4978.9  825.32  4979.4  824.82  4983.1  824.82  4983.5  825.32  4991.5  827.45
  5001.7  827.24  5010.8  828.65  5015.9  829.85  5022.1  833.06  5042.6  836.70
  5060.7  838.45  5083.4  839.81  5110.6  840.71  5115.7  841.51  5136.5  842.65
#Mann=3,-1,0
  4630.5    0.05       0  4978.9   0.033       0  4983.5    0.05       0
Bank Sta=4978.9,4983.5
Exp/Cntr=0.3,0.1

Type RM Length L Ch R = 1,13044,437,437,437
BEGIN DESCRIPTION:
Mapping XS db2749b5
END DESCRIPTION:
XS GIS Cut Line= 2
      2303327.96      7089188.44      2303831.93      7088721.84
#Sta/Elev= 30
  4582.2  836.49  4652.4  835.52  4702.2  833.37  4709.1  834.56  4758.9  831.93
  4879.1  828.32  4914.3  828.68  4921.7  829.97  4928.5  832.58  4942.6  833.25
  4950.0  830.62  4956.8  830.73  4964.2  826.99  4971.0  826.66  4978.3  821.21
  4985.2  821.14  4992.5  819.88  5018.0  819.62  5018.5  819.12  5022.6  819.62
  5034.5  820.08  5048.7  823.02  5070.2  831.06  5077.0  832.90  5105.4  838.34
  5133.7  841.69  5232.9  848.48  5253.9  851.34  5261.3  851.31  5269.0  852.32
#Mann=3,-1,0
  4582.2    0.05       0  5018.0   0.033       0  5022.6    0.05       0
Bank Sta=5018,5022.6
Exp/Cntr=0.3,0.1

Type RM Length L Ch R = 1,12607,82,82,82
BEGIN DESCRIPTION:
Mapping XS 673fa076
END DESCRIPTION:
XS GIS Cut Line= 4
      2303652.25      7089380.13      2303773.03      7089327.28
      2303802.16      7089154.43      2303828.92      7088854.44
#Sta/Elev= 30
  4761.6  830.74  4779.9  830.61  4797.8  829.31  4812.6  829.26  4844.6  827.88
  4850.0  828.10  4856.3  827.26  4873.4  826.41  4921.1  825.24  4931.2  825.71
  4951.5  825.32  4971.8  824.24  4981.9  824.42  4992.1  823.89  5002.2  820.59
  5010.0  820.02  5010.5  819.52  5014.2  819.52  5014.7  820.02  5018.5  821.32
  5042.8  822.52  5133.4  823.67  5193.6  825.87  5205.4  826.81  5213.7  829.67
  5223.8  831.74  5284.0  835.06  5344.2  840.27  5364.3  840.82  5369.9  841.52
#Mann=3,-1,0
  4761.6    0.05       0  5010.0   0.033       0  5014.7    0.05       0
Bank Sta=5010,5014.7
Exp/Cntr=0.3,0.1

Type RM Length L Ch R = 1,12525,368,368,368
BEGIN DESCRIPTION:
Mapping XS fa88d7ce
END DESCRIPTION:
XS GIS Cut Line= 4
      2303673.45      7089445.28      2303867.69      7089332.59
      2303870.56      7089057.75      2303916.37      7088856.93
#Sta/Elev= 30
  4691.0  830.11  4750.4  827.45  4756.2  827.59  4771.9  827.08  4778.3  826.48
  4824.6  825.12  4830.7  824.45  4852.2  823.82  4868.0  822.50  4873.8  822.58
  4889.5  821.76  4978.2  821.55  4988.2  821.34  5005.8  819.96  5006.3  819.46
  5010.0  819.46  5010.5  819.96  5028.2  821.99  5078.2  822.23  5118.2  823.31
  5158.2  824.96  5186.8  827.79  5190.4  827.79  5204.7  830.39  5209.8  832.22
  5247.7  835.00  5252.8  836.53  5290.7  837.24  5321.5  838.59  5396.4  843.36
#Mann=3,-1,0
  4691.0    0.05       0  5005.8   0.033       0  5010.5    0.05       0
Bank Sta=5005.8,5010.5
Exp/Cntr=0.3,0.1

Type RM Length L Ch R = 1,12157,177,177,177
BEGIN DESCRIPTION:
Mapping XS 2766252a
END DESCRIPTION:
XS GIS Cut Line= 2
      2303604.36      7089606.89      2304071.38      7089533.84
#Sta/Elev= 30
  4620.8  829.72  4631.8  829.35  4655.9  829.54  4666.0  828.36  4699.6  827.79
  4706.5  827.12  4762.3  824.16  4777.3  823.93  4807.7  822.82  4817.8  822.07
  4878.5  820.60  4898.8  820.82  4908.9  819.07  4929.1  818.77  4960.6  819.00
  4979.8  818.37  4989.9  817.90  4997.6  816.04  4998.1  815.54  5001.8  815.54
  5002.3  816.04  5010.1  817.81  5023.3  818.83  5030.4  822.81  5040.5  826.52
  5050.6  828.56  5060.7  828.83  5086.0  828.67  5089.8  828.21  5093.5  828.21
#Mann=3,-1,0
  4620.8    0.05       0  4997.6   0.033       0  5002.3    0.05       0
Bank Sta=4997.6,5002.3
Exp/Cntr=0.3,0.1

Type RM Length L Ch R = 1,11980,615,615,615
BEGIN DESCRIPTION:
MDW T 049 25.0
END DESCRIPTION:
XS GIS Cut Line= 3
      2303011.54      7090280.40      2303990.36      7089718.50
      2304379.01      7089460.00
#Sta/Elev= 30
  3884.5  838.56  3975.7  836.77  4074.0  832.44  4101.3  834.14  4138.7  834.30
  4455.0  829.02  4482.4  829.62  4550.3  827.83  4665.6  827.08  4907.8  818.24
  4981.4  818.16  4988.5  817.85  4997.2  814.29  5002.9  814.83  5007.1  812.39
  5007.6  811.89  5011.8  812.39  5015.3  812.39  5018.5  814.07  5024.5  814.21
  5033.5  819.88  5039.5  820.19  5054.6  827.56  5090.6  827.92  5147.7  825.92
  5213.9  821.56  5249.9  820.27  5299.7  823.56  5349.1  830.84  5479.9  836.65
#Mann=3,-1,0
  3884.5    0.05       0  5007.1   0.033       0  5011.8    0.05       0
Bank Sta=5007.1,5011.8
Exp/Cntr=0.3,0.1

Type RM Length L Ch R = 1,11365,409,409,409
BEGIN DESCRIPTION:
Mapping XS 506349d6
END DESCRIPTION:
XS GIS Cut Line= 2
      2304390.43      7090355.25      2304377.21      7089528.36
#Sta/Elev= 30
  4555.8  824.40  4651.1  822.36  4711.1  820.21  4751.1  820.46  4801.1  820.06
  4841.1  819.34  4901.1  816.97  4921.1  816.76  4931.1  815.95  4941.1  812.53
  4951.1  811.69  4962.2  811.36  4981.1  812.79  4991.1  812.97  4998.7  809.42
  4999.3  808.92  5003.0  808.92  5003.6  809.42  5011.1  812.27  5021.1  812.65
  5081.1  813.51  5091.1  813.23  5111.1  813.49  5201.1  816.61  5221.1  818.45
  5231.1  818.91  5261.1  822.47  5301.1  829.67  5331.1  831.56  5382.8  833.77
#Mann=3,-1,0
  4555.8    0.05       0  4998.7   0.033       0  5003.6    0.05       0
Bank Sta=4998.7,5003.6
Exp/Cntr=0.3,0.1

Type RM Length L Ch R = 1,10956,488,488,488
BEGIN DESCRIPTION:
MDW T 049 23.0
END DESCRIPTION:
XS GIS Cut Line= 3
      2304772.81      7090401.72      2304718.84      7089759.50
      2304665.64      7089423.46
#Sta/Elev= 30
  4366.5  825.34  4548.9  818.76  4587.6  816.87  4592.6  817.10  4707.5  812.83
  4859.9  810.43  4940.2  809.82  4947.3  809.38  4980.4  810.54  4990.4  806.37
  4997.9  804.75  4998.5  804.25  5002.3  804.25  5003.0  804.75  5008.2  807.16
  5013.3  807.16  5020.6  809.49  5030.7  813.81  5038.8  819.30  5051.0  821.12
  5071.2  823.17  5101.2  825.36  5111.7  826.71  5142.1  828.00  5162.3  828.25
  5173.7  829.24  5231.0  830.20  5236.0  830.70  5293.3  832.18  5351.2  834.78
#Mann=3,-1,0
  4366.5    0.05       0  4997.9   0.033       0  5003.0    0.05       0
Bank Sta=4997.9,5003
Exp/Cntr=0.3,0.1

Type RM Length L Ch R = 1,10468,466,466,466
BEGIN DESCRIPTION:
Mapping XS 438a9bf3
END DESCRIPTION:
XS GIS Cut Line= 2
      2305115.10      7090228.66      2305009.63      7089533.92
#Sta/Elev= 30
  4660.3  819.16  4866.9  813.88  4901.7  813.34  4921.9  813.68  4935.6  812.82
  4952.3  810.43  4962.4  809.91  4972.5  808.10  4982.6  803.34  4990.2  801.30
  4990.8  800.80  4994.6  800.80  4995.3  801.30  4997.6  801.62  5004.3  802.63
  5013.0  805.04  5023.1  807.00  5124.2  807.49  5195.0  810.06  5205.4  811.12
  5235.5  812.70  5245.6  813.51  5255.7  816.57  5264.0  818.10  5269.1  818.23
  5275.9  819.37  5296.2  820.92  5332.7  825.40  5345.9  825.58  5363.0  826.69
#Mann=5,-1,0
  4660.3    0.05       0  4990.2    0.07       0  4995.3    0.05       0
  4997.6    0.12       0  5345.9    0.05       0
Bank Sta=4990.2,4995.3
Exp/Cntr=0.3,0.1

Type RM Length L Ch R = 1,10002,560,560,560
BEGIN DESCRIPTION:
MDW T 049 21.0
END DESCRIPTION:
XS GIS Cut Line= 4
      2305270.21      7090441.88      2305429.93      7089929.71
      2305429.00      7089610.00      2305378.58      7089273.06
#Sta/Elev= 30
  4167.6  825.23  4318.1  820.59  4415.6  814.99  4525.7  811.67  4903.9  804.39
  4923.8  804.39  4943.8  805.36  4963.8  802.89  4983.8  801.72  4993.8  799.73
  5011.2  798.89  5011.9  798.39  5016.4  798.89  5021.3  799.72  5053.3  799.77
  5058.4  800.95  5064.3  801.25  5074.4  800.73  5084.5  802.08  5094.6  805.27
  5114.8  814.02  5127.6  817.58  5145.1  826.73  5165.4  834.19  5175.5  839.96
  5185.6  843.11  5204.7  846.43  5236.1  850.06  5266.5  852.17  5364.5  853.30
#Mann=5,-1,0
  4167.6    0.05       0  4903.9    0.12       0  5011.2    0.07       0
  5016.4    0.12       0  5204.7    0.05       0
Bank Sta=5011.2,5016.4
Exp/Cntr=0.3,0.1

Type RM Length L Ch R = 1,9442,471,471,471
BEGIN DESCRIPTION:
MDW T 049 20.0
END DESCRIPTION:
XS GIS Cut Line= 3
      2305513.26      7090403.68      2305877.88      7089709.89
      2306061.86      7089485.29
#Sta/Elev= 30
  4229.1  815.86  4278.9  813.70  4427.5  809.34  4592.6  806.16  4835.1  799.15
  4879.2  798.46  4917.6  799.60  4945.3  797.81  4961.7  797.40  4967.9  798.01
  4978.1  798.30  4983.8  797.78  4992.5  795.72  5005.8  794.26  5007.3  793.32
  5008.1  792.82  5012.6  793.32  5016.0  793.32  5020.9  795.25  5027.3  800.15
  5035.2  803.85  5041.7  808.84  5056.0  814.08  5063.9  814.63  5070.4  815.97
  5084.7  816.28  5091.2  817.49  5127.8  818.96  5134.3  819.76  5303.2  826.33
#Mann=5,-1,0
  4229.1    0.05       0  4967.9    0.12       0  4992.5    0.05       0
  5007.3   0.033       0  5012.6    0.05       0
Bank Sta=5007.3,5012.6
Exp/Cntr=0.3,0.1

Type RM Length L Ch R = 1,8971,400,400,400
BEGIN DESCRIPTION:
MDW T 049 19.0
END DESCRIPTION:
XS GIS Cut Line= 3
      2305827.50      7090488.31      2306072.24      7090103.52
      2306238.40      7089593.32
#Sta/Elev= 30
  4550.1  808.76  4679.2  805.44  4724.9  805.06  4803.7  801.76  4927.3  798.79
  4949.3  797.28  4955.2  796.02  4985.7  795.56  4998.4  788.58  5002.6  788.44
  5003.4  787.94  5007.9  788.44  5020.3  793.57  5050.4  794.62  5135.9  794.49
  5167.6  797.07  5188.6  800.68  5199.1  803.28  5205.0  806.10  5230.7  809.93
  5236.9  812.81  5251.7  815.99  5277.5  819.12  5314.8  822.12  5428.4  827.86
  5472.6  829.24  5492.3  830.88  5497.5  830.42  5524.2  831.67  5542.7  830.93
#Mann=5,-1,0
  4550.1    0.05       0  5002.6   0.033       0  5007.9    0.05       0
  5050.4    0.12       0  5277.5    0.05       0
Bank Sta=5002.6,5007.9
Exp/Cntr=0.3,0.1

Type RM Length L Ch R = 1,8571,295,295,295
BEGIN DESCRIPTION:
MDW T 049 18.0
END DESCRIPTION:
XS GIS Cut Line= 3
      2306463.76      7090643.62      2306459.05      7090130.12
      2306330.09      7089659.28
#Sta/Elev= 30
  4488.2  808.88  4531.8  807.74  4711.8  799.06  4801.8  796.18  4861.8  795.10
  4881.8  795.24  4901.8  794.24  4971.8  792.64  4981.8  790.63  4996.6  785.05
  4997.4  784.55  5001.2  784.55  5002.0  785.05  5012.2  786.58  5019.1  789.96
  5038.3  790.30  5093.3  790.13  5126.3  791.29  5178.1  795.12  5198.8  797.23
  5212.2  799.11  5219.6  801.79  5233.7  804.63  5281.2  810.59  5292.2  812.59
  5326.1  814.89  5365.7  817.04  5426.9  819.26  5439.9  820.28  5489.9  821.62
#Mann=5,-1,0
  4488.2    0.05       0  4996.6   0.033       0  5002.0    0.05       0
  5038.3    0.12       0  5233.7    0.05       0
Bank Sta=4996.6,5002
Exp/Cntr=0.3,0.1

Type RM Length L Ch R = 1,8276,437,437,437
BEGIN DESCRIPTION:
MDW T 049 17.0
END DESCRIPTION:
XS GIS Cut Line= 3
      2306930.81      7090464.02      2306727.15      7090016.24
      2306549.71      7089607.18
#Sta/Elev= 30
  4513.5  806.55  4532.2  805.90  4555.2  803.80  4561.9  801.56  4578.3  799.70
  4583.8  798.27  4665.6  790.68  4693.6  789.03  4745.2  787.71  4894.6  787.73
  4963.3  787.61  4979.3  787.33  4986.8  781.93  4997.9  780.77  4998.7  780.27
  5003.3  780.77  5005.4  780.77  5015.5  785.13  5023.1  785.94  5044.9  787.15
  5058.7  786.39  5085.9  786.00  5109.4  791.00  5290.0  801.73  5360.4  804.02
  5365.8  805.01  5418.2  806.27  5436.2  805.93  5441.6  807.05  5451.3  807.14
#Mann=7,-1,0
  4513.5    0.05       0  4665.6    0.12       0  4894.6    0.05       0
  4963.3    0.12       0  4997.9    0.07       0  5003.3    0.12       0
  5058.7    0.05       0
Bank Sta=4997.9,5003.3
Exp/Cntr=0.3,0.1

Type RM Length L Ch R = 1,7839,561,561,561
BEGIN DESCRIPTION:
MDW T 049 16.0
END DESCRIPTION:
XS GIS Cut Line= 3
      2307076.63      7090436.22      2307098.99      7089910.03
      2307114.77      7089503.60
#Sta/Elev= 30
  4471.0  801.32  4537.3  798.51  4557.3  796.92  4627.4  793.78  4657.4  791.36
  4677.4  788.72  4697.4  787.07  4757.5  783.73  4807.9  782.36  4867.6  781.78
  4887.6  780.90  4957.7  781.10  4977.7  778.56  4992.4  773.33  4993.2  772.83
  4997.1  772.83  4998.0  773.33  5007.7  774.48  5017.7  777.68  5027.7  780.09
  5057.7  784.36  5124.8  788.40  5135.8  788.65  5177.8  791.83  5227.9  794.46
  5317.9  801.53  5378.0  806.65  5383.7  807.86  5398.0  808.92  5404.4  809.99
#Mann=5,-1,0
  4471.0    0.05       0  4807.9    0.12       0  4992.4    0.07       0
  4998.0    0.12       0  5135.8    0.05       0
Bank Sta=4992.4,4998
Exp/Cntr=0.3,0.1

Type RM Length L Ch R = 1,7278,348,348,348
BEGIN DESCRIPTION:
MDW T 049 15.0
END DESCRIPTION:
XS GIS Cut Line= 3
      2307453.37      7090438.83      2307608.82      7089859.74
      2307640.01      7089575.94
#Sta/Elev= 30
  4400.4  793.35  4533.8  788.24  4553.2  786.49  4558.4  786.93  4575.2  785.64
  4598.4  785.39  4658.0  781.81  4713.2  775.56  4757.4  775.10  4782.3  774.12
  4788.0  774.94  4822.8  775.40  4968.7  774.50  4982.8  771.82  4989.4  769.17
  4994.5  768.77  4995.3  768.27  5000.1  768.77  5009.8  769.25  5019.9  774.22
  5046.2  781.40  5080.2  785.49  5102.7  787.28  5137.2  790.71  5150.6  790.94
  5180.8  793.78  5190.9  795.60  5228.3  799.31  5241.2  799.24  5285.5  803.01
#Mann=5,-1,0
  4400.4    0.05       0  4757.4    0.12       0  4994.5    0.07       0
  5000.1    0.12       0  5102.7    0.05       0
Bank Sta=4994.5,5000.1
Exp/Cntr=0.3,0.1

Type RM Length L Ch R = 1,6930,314,314,314
BEGIN DESCRIPTION:
MDW T 049 14.0
END DESCRIPTION:
XS GIS Cut Line= 3
      2307830.10      7090460.56      2307891.78      7089959.91
      2307895.21      7089507.36
#Sta/Elev= 30
  4506.7  787.83  4658.4  783.26  4809.5  777.04  4839.8  775.11  4859.9  773.31
  4880.1  770.75  4930.4  769.38  4946.5  769.97  4951.6  769.70  4960.7  770.69
  4980.8  770.18  4990.9  768.79  4998.1  765.05  4999.0  764.55  5002.9  764.55
  5003.8  765.05  5008.6  766.31  5021.1  766.69  5051.1  769.37  5091.1  769.92
  5101.1  772.23  5121.7  774.55  5151.1  778.78  5161.1  779.81  5171.1  780.26
  5191.1  782.28  5222.4  783.85  5371.1  790.87  5421.1  794.71  5463.7  796.82
#Mann=5,-1,0
  4506.7    0.05       0  4998.1   0.033       0  5003.8    0.05       0
  5121.7    0.12       0  5222.4    0.05       0
Bank Sta=4998.1,5003.8
Exp/Cntr=0.3,0.1

Type RM Length L Ch R = 1,6616,492,492,492
BEGIN DESCRIPTION:
Mapping XS 7b00a767
END DESCRIPTION:
XS GIS Cut Line= 4
      2307879.54      7090417.89      2307930.09      7090115.41
      2308163.71      7090070.26      2308127.52      7089856.62
#Sta/Elev= 30
  4622.2  784.80  4691.0  783.35  4731.6  781.87  4762.0  781.24  4829.6  778.13
  4883.7  776.12  4914.1  773.35  4924.0  771.58  4928.9  771.58  4931.9  770.43
  4958.3  768.90  4978.7  763.61  4983.8  764.40  4988.9  762.31  4996.2  760.79
  4997.1  760.29  5001.0  760.29  5001.9  760.79  5009.2  762.62  5019.4  764.48
  5040.7  765.53  5087.4  765.63  5121.3  767.06  5144.3  767.31  5169.5  767.01
  5207.7  767.93  5248.2  769.77  5284.3  770.26  5289.3  769.88  5383.5  772.19
#Mann=3,-1,0
  4622.2    0.05       0  4996.2   0.033       0  5001.9    0.05       0
Bank Sta=4996.2,5001.9
Exp/Cntr=0.3,0.1

Type RM Length L Ch R = 1,6124,315,315,315
BEGIN DESCRIPTION:
Mapping XS 4e49cfca
END DESCRIPTION:
XS GIS Cut Line= 3
      2308221.26      7090438.67      2308347.57      7090378.83
      2308355.35      7089929.17
#Sta/Elev= 30
  4720.7  771.41  4732.0  770.76  4762.5  768.24  4772.0  766.64  4777.5  766.36
  4800.3  763.48  4806.7  761.97  4817.5  760.82  4845.8  760.43  4879.3  761.15
  4909.3  761.08  4949.3  759.18  4979.3  756.61  4986.3  755.70  4987.3  755.20
  4991.4  755.20  4992.4  755.70  5009.3  757.60  5019.3  759.30  5029.3  763.37
  5075.9  763.54  5109.3  764.69  5169.3  764.98  5209.4  765.99  5233.2  766.12
  5249.4  766.93  5259.4  766.78  5269.4  767.31  5289.4  767.74  5310.2  769.03
#Mann=4,-1,0
  4720.7    0.05       0  4986.3   0.033       0  4992.4    0.05       0
  5075.9    0.12       0
#XS Ineff=2,0
    0.00 4895.60  766.09               0
Permanent Ineff=
       F       F
Bank Sta=4986.3,4992.4
Exp/Cntr=0.3,0.1

Type RM Length L Ch R = 1,5809,125,125,125
BEGIN DESCRIPTION:
Mapping XS 13248a72
END DESCRIPTION:
XS GIS Cut Line= 4
      2308198.57      7090580.55      2308493.23      7090491.90
      2308681.40      7090162.88      2308765.36      7090110.68
#Sta/Elev= 30
  4545.6  773.01  4619.1  768.13  4634.5  768.69  4705.8  765.36  4744.5  758.77
  4765.3  759.20  4771.8  760.34  4777.1  758.42  4804.9  760.02  4879.7  757.42
  4970.3  758.42  4982.2  757.93  4997.7  754.70  5013.5  753.45  5028.3  754.93
  5050.9  755.52  5097.5  755.23  5137.3  756.37  5177.4  750.98  5178.4  750.48
  5183.6  750.98  5189.6  754.96  5202.1  759.78  5262.6  762.57  5299.2  771.50
  5305.1  772.06  5311.9  776.10  5320.4  778.86  5326.3  777.72  5331.2  780.07
#Mann=4,-1,0
  4545.6    0.05       0  5097.5    0.12       0  5177.4   0.033       0
  5183.6    0.12       0
#XS Ineff=1,-1
 4635.10 4954.50  764.29
Permanent Ineff=
       F
Bank Sta=5177.4,5183.6
Exp/Cntr=0.3,0.1

Type RM Length L Ch R = 1,5684,440,440,440
BEGIN DESCRIPTION:
MDW T 049 12.0
END DESCRIPTION:
XS GIS Cut Line= 3
      2308129.05      7090635.70      2308623.21      7090462.35
      2308961.14      7090413.66
#Sta/Elev= 30
  4481.0  778.13  4618.7  770.44  4660.1  766.96  4696.4  766.46  4745.9  764.24
  4758.4  762.58  4777.7  762.47  4877.1  758.51  4926.0  756.23  4933.8  755.11
  4939.1  755.89  4964.8  752.90  4970.1  754.24  4997.6  749.03  4998.6  748.53
  5003.8  749.03  5020.6  750.65  5030.7  753.89  5046.7  753.99  5061.2  754.01
  5091.4  760.05  5121.5  770.50  5126.5  769.45  5131.8  774.40  5152.0  782.07
  5162.1  783.25  5232.8  786.10  5250.2  788.50  5283.3  793.31  5346.1  797.94
#Mann=5,-1,0
  4481.0    0.05       0  4997.6   0.033       0  5003.8    0.05       0
  5046.7    0.12       0  5250.2    0.05       0
Bank Sta=4997.6,5003.8
Exp/Cntr=0.3,0.1

Type RM Length L Ch R = 1,5244,424,424,424
BEGIN DESCRIPTION:
MDW T 049 11.0
END DESCRIPTION:
XS GIS Cut Line= 3
      2308153.06      7090812.09      2308477.97      7090804.58
      2308925.68      7090764.49
#Sta/Elev= 30
  4675.0  780.50  4710.5  777.56  4731.0  775.46  4841.0  768.27  4881.0  764.76
  4931.0  761.46  4971.0  757.55  4979.0  748.92  4984.0  749.28  4994.9  742.37
  4995.9  741.87  5001.2  742.37  5031.2  746.70  5071.3  749.90  5101.4  750.32
  5141.6  751.85  5171.7  754.70  5211.9  757.11  5232.0  759.13  5252.0  762.83
  5282.2  764.61  5322.3  768.36  5334.5  770.15  5382.6  779.95  5392.6  782.49
  5412.7  786.19  5432.8  790.46  5440.8  792.76  5445.8  793.28  5449.5  794.76
#Mann=4,-1,0
  4675.0    0.05       0  4710.5    0.12       0  4994.9   0.033       0
  5001.2    0.05       0
Bank Sta=4994.9,5001.2
Exp/Cntr=0.3,0.1

Type RM Length L Ch R = 1,4820,526,526,526
BEGIN DESCRIPTION:
MDW T 049 10.0
END DESCRIPTION:
XS GIS Cut Line= 3
      2308200.74      7091156.71      2308628.89      7091170.05
      2309155.72      7091174.05
#Sta/Elev= 30
  4566.1  795.72  4584.4  792.46  4604.4  790.56  4714.4  782.72  4734.4  778.27
  4764.5  768.40  4790.3  762.90  4824.5  761.10  4844.5  758.86  4884.5  757.14
  4924.5  751.98  4934.5  749.52  4964.5  745.19  4984.6  743.50  4992.0  741.17
  5011.4  738.62  5012.4  738.12  5017.7  738.62  5044.6  747.58  5164.6  754.22
  5254.6  761.53  5284.6  762.84  5344.6  769.77  5372.5  774.61  5384.6  776.32
  5414.6  777.89  5434.6  780.59  5454.6  783.61  5474.6  789.10  5521.3  796.48
#Mann=5,-1,0
  4566.1    0.05       0  4790.3    0.12       0  5011.4    0.07       0
  5017.7    0.12       0  5372.5    0.05       0
Bank Sta=5011.4,5017.7
Exp/Cntr=0.3,0.1

Type RM Length L Ch R = 1,4294,366,366,366
BEGIN DESCRIPTION:
MDW T 049 9.0
END DESCRIPTION:
XS GIS Cut Line= 3
      2308250.21      7091695.77      2308879.77      7091599.37
      2309202.55      7091577.71
#Sta/Elev= 30
  4381.8  785.39  4400.8  781.12  4461.5  772.60  4491.9  769.49  4518.1  765.12
  4600.6  757.24  4713.3  746.38  4815.6  742.41  4845.1  740.38  4876.3  739.58
  4896.5  740.20  4918.6  739.23  4947.1  739.98  4997.7  736.67  5004.6  735.19
  5005.7  734.69  5011.0  735.19  5020.8  735.54  5038.0  744.78  5048.0  747.32
  5068.0  755.49  5178.3  767.74  5208.4  772.81  5218.4  776.21  5233.4  779.13
  5238.4  781.11  5254.5  784.01  5268.5  785.31  5308.6  793.18  5342.2  797.33
#Mann=5,-1,0
  4381.8    0.05       0  4600.6    0.12       0  5004.6    0.07       0
  5011.0    0.12       0  5254.5    0.05       0
Bank Sta=5004.6,5011
Exp/Cntr=0.3,0.1

Type RM Length L Ch R = 1,3928,480,480,480
BEGIN DESCRIPTION:
MDW T 049 8.0
END DESCRIPTION:
XS GIS Cut Line= 3
      2308308.41      7091911.91      2308871.97      7091859.79
      2309213.81      7091843.34
#Sta/Elev= 30
  4427.8  785.22  4468.6  782.62  4478.6  780.26  4514.1  775.35  4548.9  770.17
  4569.0  765.85  4589.1  764.74  4607.8  762.39  4612.8  762.77  4659.4  753.67
  4722.3  747.89  4749.8  742.98  4779.9  740.07  4840.1  739.27  4880.3  736.86
  4920.5  736.97  4936.4  732.95  4960.7  735.19  4980.7  735.41  5007.6  732.36
  5008.6  731.86  5014.0  732.36  5030.8  743.45  5089.7  748.00  5131.0  752.58
  5251.1  769.61  5290.5  776.52  5298.8  778.83  5321.2  781.94  5336.0  782.84
#Mann=5,-1,0
  4427.8    0.05       0  4514.1    0.12       0  5007.6    0.07       0
  5014.0    0.12       0  5290.5    0.05       0
Bank Sta=5007.6,5014
Exp/Cntr=0.3,0.1

Type RM Length L Ch R = 1,3448,469,469,469
BEGIN DESCRIPTION:
MDW T 049 7.0
END DESCRIPTION:
XS GIS Cut Line= 3
      2308282.39      7092252.19      2308878.28      7092249.29
      2309374.17      7092252.19
#Sta/Elev= 30
  4404.1  784.74  4440.7  781.71  4460.7  776.84  4473.2  775.08  4530.7  767.31
  4590.7  762.03  4680.7  750.28  4700.7  746.34  4750.7  740.50  4860.7  735.82
  4900.7  733.16  4940.7  733.64  4970.7  728.98  4994.6  728.09  4995.7  727.59
  5001.1  728.09  5002.9  728.09  5010.7  733.89  5020.7  735.62  5054.9  736.76
  5100.7  738.66  5140.7  747.50  5160.7  749.74  5250.7  752.49  5310.7  767.24
  5350.7  772.83  5380.7  778.64  5410.7  782.03  5490.7  788.73  5495.9  791.05
#Mann=5,-1,0
  4404.1    0.05       0  4473.2    0.12       0  4994.6    0.07       0
  5001.1    0.12       0  5054.9    0.05       0
Bank Sta=4994.6,5001.1
Exp/Cntr=0.3,0.1

Type RM Length L Ch R = 1,2979,504,504,504
BEGIN DESCRIPTION:
MDW T 049 6.0
END DESCRIPTION:
XS GIS Cut Line= 3
      2308225.08      7092578.58      2308929.50      7092634.82
      2309390.02      7092656.71
#Sta/Elev= 30
  4274.8  786.13  4329.6  782.27  4354.7  773.50  4389.1  769.37  4409.1  765.45
  4459.3  762.23  4519.5  754.27  4559.6  751.93  4619.8  742.58  4700.1  733.31
  4840.5  730.06  4910.7  730.91  4950.9  729.00  4973.6  726.15  4985.6  725.61
  4987.7  724.36  4988.7  723.86  4994.3  724.36  5001.0  724.84  5021.0  731.23
  5041.0  739.96  5071.1  746.41  5141.1  754.26  5191.1  761.64  5196.1  761.16
  5201.2  762.83  5241.3  766.26  5311.3  779.63  5361.4  783.45  5442.5  786.40
#Mann=5,-1,0
  4274.8    0.05       0  4329.6    0.12       0  4973.6    0.05       0
  4987.7   0.033       0  4994.3    0.05       0
Bank Sta=4987.7,4994.3
Exp/Cntr=0.3,0.1

Type RM Length L Ch R = 1,2475,321,321,321
BEGIN DESCRIPTION:
MDW T 049 5.0
END DESCRIPTION:
XS GIS Cut Line= 3
      2308116.52      7092840.73      2308686.77      7092866.12
      2309331.83      7092883.27
#Sta/Elev= 30
  4433.7  778.97  4460.5  779.95  4525.5  781.22  4546.3  778.61  4576.3  772.91
  4616.4  767.57  4636.4  766.98  4676.4  762.84  4746.5  757.59  4766.5  753.61
  4826.6  746.89  4856.6  742.19  4906.7  737.41  4946.7  732.40  4996.7  728.59
  4999.8  720.11  5000.9  719.61  5006.4  720.11  5016.8  720.24  5066.8  726.96
  5156.8  729.25  5206.8  729.28  5266.8  731.89  5335.3  741.56  5340.3  740.95
  5446.9  757.00  5496.9  762.11  5539.8  769.74  5576.9  779.42  5649.8  782.51
#Mann=5,-1,0
  4433.7    0.05       0  4460.5    0.12       0  4999.8    0.07       0
  5006.4    0.12       0  5539.8    0.05       0
Bank Sta=4999.8,5006.4
Exp/Cntr=0.3,0.1

Type RM Length L Ch R = 1,2154,587,587,587
BEGIN DESCRIPTION:
MDW T 049 4.0
END DESCRIPTION:
XS GIS Cut Line= 3
      2308163.54      7093091.33      2308825.91      7093118.31
      2309222.83      7093125.28
#Sta/Elev= 30
  4346.2  760.84  4391.7  762.06  4491.8  758.38  4541.8  752.15  4742.0  737.94
  4832.1  728.40  4872.1  726.49  4922.1  725.53  4952.2  723.40  4962.2  723.66
  4982.2  720.38  5002.2  718.74  5008.2  717.05  5018.9  716.48  5019.9  715.98
  5025.6  716.48  5032.2  721.01  5042.2  725.45  5062.2  726.52  5082.2  731.03
  5162.2  740.14  5172.2  742.54  5222.2  750.33  5272.3  759.53  5302.3  761.49
  5312.3  763.37  5332.3  763.56  5388.6  772.26  5402.6  773.23  5406.1  773.23
#Mann=4,-1,0
  4346.2    0.12       0  5018.9    0.07       0  5025.6    0.12       0
  5402.6    0.05       0
Bank Sta=5018.9,5025.6
Exp/Cntr=0.3,0.1

Type RM Length L Ch R = 1,1567,101,101,101
BEGIN DESCRIPTION:
Mapping XS 7439bf51
END DESCRIPTION:
XS GIS Cut Line= 2
      2308130.97      7093520.78      2309168.92      7093467.69
#Sta/Elev= 30
  4408.8  772.58  4567.0  762.28  4637.1  754.36  4714.9  749.29  4757.3  739.57
  4777.3  737.94  4797.3  734.73  4807.3  730.59  4817.4  724.94  4827.4  721.60
  4837.4  720.37  4857.4  719.71  4927.5  720.56  4987.6  712.91  4997.6  713.20
  5014.3  711.75  5015.3  711.25  5021.0  711.75  5027.6  713.07  5037.6  719.28
  5047.7  722.71  5090.6  722.60  5129.7  722.90  5167.8  723.84  5227.9  730.44
  5288.0  739.65  5368.1  755.37  5388.1  758.42  5418.1  760.94  5448.1  767.42
#Mann=5,-1,0
  4408.8    0.12       0  5014.3    0.07       0  5021.0    0.12       0
  5090.6    0.05       0  5129.7    0.12       0
Bank Sta=5014.3,5021
Exp/Cntr=0.3,0.1

Type RM Length L Ch R = 1,1466,681,681,681
BEGIN DESCRIPTION:
MDW T 049 3.0
END DESCRIPTION:
XS GIS Cut Line= 3
      2308135.74      7093612.16      2308679.29      7093585.12
      2309184.20      7093572.23
#Sta/Elev= 30
  4425.9  769.81  4549.3  762.26  4567.2  759.64  4572.2  761.16  4589.4  757.69
  4619.4  754.54  4709.5  747.56  4767.9  734.77  4772.9  735.18  4789.6  732.87
  4879.7  716.11  4908.8  717.64  4939.8  719.50  4949.8  718.78  4959.8  716.41
  4967.5  711.19  4986.5  709.90  4987.5  709.40  4993.2  709.90  5009.8  711.72
  5019.9  717.76  5029.9  720.25  5083.0  721.24  5179.9  722.32  5239.9  728.62
  5330.0  743.26  5390.0  755.53  5420.0  758.89  5470.0  768.52  5475.2  770.45
#Mann=5,-1,0
  4425.9    0.12       0  4908.8    0.05       0  4986.5   0.033       0
  4993.2    0.05       0  5083.0    0.12       0
Bank Sta=4986.5,4993.2
Exp/Cntr=0.3,0.1

Type RM Length L Ch R = 1,785,214,214,214
BEGIN DESCRIPTION:
MDW T 049 2.0
END DESCRIPTION:
XS GIS Cut Line= 3
      2308007.23      7093681.58      2308384.10      7094004.53
      2309178.98      7093710.01
#Sta/Elev= 30
  4501.6  775.07  4728.2  757.59  4771.0  749.30  4825.8  742.83  4877.5  738.76
  4913.5  738.44  4941.1  733.82  4948.8  723.55  4955.4  729.09  4963.1  704.84
  4969.7  709.13  4977.4  704.30  4987.8  703.63  4988.9  703.13  4994.6  703.63
  4997.8  705.88  5027.6  711.48  5058.0  714.17  5440.4  717.75  5517.5  720.72
  5542.6  725.77  5603.3  732.48  5628.4  738.14  5633.7  737.35  5719.5  749.44
  5744.6  754.88  5775.0  757.34  5805.4  762.88  5830.4  771.57  5845.6  774.55
#Mann=5,-1,0
  4501.6    0.12       0  4825.8    0.05       0  4913.5    0.12       0
  4987.8    0.07       0  4994.6    0.12       0
Bank Sta=4987.8,4994.6
Exp/Cntr=0.3,0.1
