--- Morris Branch.prj (project) ---

Proj Title=Morris Branch Base Level Engineering
Current Plan=p01
Default Exp/Contr=0.3,0.1
English Units
Geom File=g01
Flow File=f01
Plan File=p01
BEGIN DESCRIPTION:
Morris Branch
END DESCRIPTION:

--- Morris Branch.p01 (plan) ---

Plan Title=Multiple Run
Short Identifier=Multiple
Geom File=g01
Flow File=f01
Subcritical Flow
K Sum by GR= 0
Std Step Tol= 0.01
Critical Tol= 0.01
Num of Std Step Trials= 20
Max Error Tol= 0.3
Flow Tol Ratio= 0.001
Split Flow NTrial= 30
Split Flow Tol= 0.02
Split Flow Ratio= 0.02
Log Output Level= 0
Friction Slope Method= 1
Unsteady Friction Slope Method= 2
Unsteady Bridges Friction Slope Method= 1
Parabolic Critical Depth
Global Vel Dist=  1 , 1 , 1
Global Log Level= 0
CheckData=True
Encroach Param= -1, 0, 0, 0
BEGIN DESCRIPTION:
Multiple Run
END DESCRIPTION:

--- Morris Branch.f01 (steady flow) ---

Flow Title=Multiple
Number of Profiles=7
Profile Names=10-year,25-year,50-year,1pct_min,100-year,1pct_plu,500-year
River Rch & RM= Morris Branch,Reach-1,58139
     470     638     776     469     937    1869    1366
River Rch & RM= Morris Branch,Reach-1,54130
     673     933    1151     705    1407    2807    2108
River Rch & RM= Morris Branch,Reach-1,53388
     686     954    1177     722    1441    2875    2163
River Rch & RM= Morris Branch,Reach-1,52975
     749    1045    1293     795    1586    3164    2390
River Rch & RM= Morris Branch,Reach-1,51228
    1042    1477    1847    1145    2284    4558    3507
River Rch & RM= Morris Branch,Reach-1,47402
    1199    1707    2141    1331    2655    5298    4098
River Rch & RM= Morris Branch,Reach-1,43192
    1332    1906    2398    1495    2983    5952    4630
River Rch & RM= Morris Branch,Reach-1,41841
    1541    2217    2800    1750    3492    6968    5453
River Rch & RM= Morris Branch,Reach-1,37012
    1727    2494    3158    1978    3947    7875    6187
River Rch & RM= Morris Branch,Reach-1,35228
    1824    2643    3353    2105    4200    8380    6612
River Rch & RM= Morris Branch,Reach-1,33091
    1987    2887    3672    2309    4608    9193    7281
River Rch & RM= Morris Branch,Reach-1,30839
    2045    2972    3779    2376    4740    9458    7486
River Rch & RM= Morris Branch,Reach-1,24526
    2695    3959    5070    3208    6400   12771   10238
River Rch & RM= Morris Branch,Reach-1,17904
    3155    4658    5987    3800    7581   15127   12201
River Rch & RM= Morris Branch,Reach-1,13442
    3401    5034    6481    4119    8219   16399   13267
River Rch & RM= Morris Branch,Reach-1,10973
    3424    5053    6493    4118    8217   16395   13207
Boundary for River Rch & Prof#=Morris Branch,Reach-1,1
Up Type=0
Dn Type=3
Dn Slope=0.005
Boundary for River Rch & Prof#=Morris Branch,Reach-1,2
Up Type=0
Dn Type=3
Dn Slope=0.005
Boundary for River Rch & Prof#=Morris Branch,Reach-1,3
Up Type=0
Dn Type=3
Dn Slope=0.005
Boundary for River Rch & Prof#=Morris Branch,Reach-1,4
Up Type=0
Dn Type=3
Dn Slope=0.005
Boundary for River Rch & Prof#=Morris Branch,Reach-1,5
Up Type=0
Dn Type=3
Dn Slope=0.005
Boundary for River Rch & Prof#=Morris Branch,Reach-1,6
Up Type=0
Dn Type=3
Dn Slope=0.005
Boundary for River Rch & Prof#=Morris Branch,Reach-1,7
Up Type=0
Dn Type=3
Dn Slope=0.005

--- Morris Branch.g01 (geometry) ---

Geom Title=Existing Conditions

River Reach=Morris Branch,Reach-1
Reach XY= 30
      2284229.00      7125960.00      2287499.16      7123640.37
      2289665.37      7120772.93      2290399.48      7120940.74
      2291326.62      7119315.37      2291973.33      7119708.02
      2295227.32      7118406.91      2295679.19      7117894.71
      2295331.90      7117467.91      2296385.09      7117152.52
      2296476.29      7116665.28      2300917.51      7115608.53
      2301934.97      7114562.14      2302084.85      7115007.94
      2303113.81      7114509.89      2305170.86      7115407.05
      2307809.21      7113080.09      2308069.32      7112320.19
      2308720.53      7112457.42      2310673.82      7111204.59
      2311022.33      7109968.96      2313017.17      7109758.38
      2313976.45      7108815.05      2315099.19      7108409.62
      2315773.33      7108708.02      2317153.88      7107759.71
      2318075.72      7108752.00      2318298.91      7108409.89
      2319470.69      7108662.97      2320029.00      7109710.00

Type RM Length L Ch R = 1,58139,279,279,279
BEGIN DESCRIPTION:
Morris Branch 109.0
END DESCRIPTION:
XS GIS Cut Line= 3
      2284629.00      7126060.00      2284429.00      7125760.00
      2284229.01      7125460.01
#Sta/Elev= 30
  4634.7  930.47  4720.3  926.94  4750.4  925.04  4756.4  925.33  4765.4  924.45
  4771.4  924.68  4786.4  923.38  4815.0  922.38  4858.5  921.63  4887.1  920.61
  4945.7  920.51  4970.7  919.99  4971.0  919.49  4974.5  919.49  4974.7  919.99
  5031.3  920.48  5044.8  920.13  5053.8  921.21  5067.4  920.36  5080.9  921.01
  5095.9  921.04  5110.9  921.88  5116.9  921.39  5126.0  922.98  5147.0  923.58
  5153.0  922.55  5168.0  923.94  5198.1  925.56  5283.7  929.07  5355.8  933.32
#Mann=3,-1,0
  4634.7    0.05       0  4970.7    0.04       0  4974.7    0.05       0
Bank Sta=4970.7,4974.7
Exp/Cntr=0.3,0.1

Type RM Length L Ch R = 1,57860,259,259,259
BEGIN DESCRIPTION:
Morris Branch 108.0
END DESCRIPTION:
XS GIS Cut Line= 3
      2284779.01      7125910.02      2284629.00      7125610.00
      2284329.00      7125310.00
#Sta/Elev= 30
  4670.7  927.29  4715.4  926.23  4768.5  923.00  4813.3  921.40  4841.2  921.13
  4849.6  920.25  4858.0  919.90  4885.9  919.86  4894.3  920.53  4902.7  919.13
  4916.7  918.74  4925.1  918.92  4939.0  916.73  4947.4  917.23  4953.0  917.96
  4997.7  916.93  5003.3  917.23  5020.3  917.07  5046.6  916.15  5046.8  915.65
  5050.3  915.65  5050.6  916.15  5076.8  916.90  5119.3  919.96  5218.3  924.16
  5260.7  927.08  5274.8  927.37  5331.4  930.05  5373.8  932.67  5430.4  934.88
#Mann=3,-1,0
  4670.7    0.05       0  5046.6   0.033       0  5050.6    0.05       0
Bank Sta=5046.6,5050.6
Exp/Cntr=0.3,0.1

Type RM Length L Ch R = 1,57601,242,242,242
BEGIN DESCRIPTION:
Morris Branch 107.0
END DESCRIPTION:
XS GIS Cut Line= 3
      2284929.01      7125760.03      2284829.00      7125460.00
      2284528.97      7125309.99
#Sta/Elev= 30
  4679.3  926.08  4682.0  926.08  4689.9  923.62  4700.4  923.20  4732.0  923.11
  4742.6  921.87  4784.7  920.79  4795.3  919.73  4879.6  917.67  4942.9  914.64
  4974.5  914.79  4985.0  913.22  4990.9  910.78  4991.2  910.28  4994.7  910.28
  4994.9  910.78  5003.9  910.88  5009.5  911.87  5017.9  914.56  5031.9  915.09
  5054.3  914.86  5093.4  915.39  5099.0  916.20  5107.4  916.21  5121.3  917.60
  5129.7  917.66  5152.1  919.20  5241.5  921.97  5286.2  923.99  5331.0  926.82
#Mann=3,-1,0
  4679.3    0.05       0  4990.9   0.033       0  4994.9    0.05       0
Bank Sta=4990.9,4994.9
Exp/Cntr=0.3,0.1

Type RM Length L Ch R = 1,57359,282,282,282
BEGIN DESCRIPTION:
Morris Branch 106.0
END DESCRIPTION:
XS GIS Cut Line= 3
      2285078.99      7125609.98      2284979.00      7125310.00
      2284678.97      7125109.98
#Sta/Elev= 30
  4678.0  923.05  4688.5  922.98  4699.1  921.52  4751.8  919.17  4762.3  918.34
  4804.5  916.94  4815.0  916.95  4846.6  915.61  4857.2  914.58  4867.7  914.56
  4888.8  913.46  4973.1  913.23  4983.7  911.29  5001.7  910.33  5007.7  909.50
  5014.7  909.14  5015.0  908.64  5018.5  908.64  5018.7  909.14  5022.8  912.89
  5030.3  913.30  5043.8  913.42  5102.4  915.52  5109.9  915.43  5138.4  916.75
  5145.9  916.44  5182.0  917.39  5210.5  919.31  5305.2  922.26  5354.8  924.66
#Mann=3,-1,0
  4678.0    0.05       0  5014.7   0.033       0  5018.7    0.05       0
Bank Sta=5014.7,5018.7
Exp/Cntr=0.3,0.1

Type RM Length L Ch R = 1,57077,153,153,153
BEGIN DESCRIPTION:
Morris Branch 105.0
END DESCRIPTION:
XS GIS Cut Line= 3
      2285129.00      7125610.00      2285179.00      7125110.00
      2285078.98      7124959.97
#Sta/Elev= 30
  4502.0  922.32  4542.2  921.45  4562.3  920.15  4612.5  917.88  4632.6  917.54
  4642.7  916.81  4750.7  913.42  4755.8  913.66  4773.3  911.40  4783.4  910.82
  4803.5  910.92  4823.6  910.44  4843.7  911.96  4883.9  910.79  4893.9  911.05
  4956.8  910.28  4984.4  909.63  5000.0  907.45  5000.2  906.95  5003.7  906.95
  5004.0  907.45  5007.5  907.45  5018.0  909.79  5063.1  909.85  5099.1  911.22
  5141.2  913.62  5162.2  915.51  5171.2  915.88  5181.8  917.46  5184.8  917.46
#Mann=3,-1,0
  4502.0    0.05       0  5000.0   0.033       0  5004.0    0.05       0
#XS Ineff=2,0
    0.00 4906.40  915.67               0
Permanent Ineff=
       F       F
Bank Sta=5000,5004
Exp/Cntr=0.3,0.1

Type RM Length L Ch R = 1,56924,415,415,415
BEGIN DESCRIPTION:
Mapping XS b6281dbc
END DESCRIPTION:
XS GIS Cut Line= 3
      2285346.63      7125481.26      2285333.57      7125145.67
      2285295.52      7124764.71
#Sta/Elev= 30
  4633.9  914.41  4755.2  912.26  4765.3  911.74  4835.3  909.91  4845.3  909.86
  4855.3  909.38  4865.3  909.44  4905.4  908.34  4969.7  908.28  4975.4  906.69
  4985.5  906.26  4995.5  908.58  5005.6  909.19  5025.7  909.48  5035.7  908.92
  5068.5  908.95  5075.9  907.99  5084.0  906.24  5084.2  905.74  5087.7  905.74
  5088.0  906.24  5096.0  909.29  5146.3  910.39  5169.0  911.24  5186.5  911.39
  5216.6  912.34  5236.7  912.68  5317.1  915.76  5347.3  916.55  5352.6  916.92
#Mann=3,-1,0
  4633.9    0.05       0  5084.0   0.033       0  5088.0    0.05       0
Bank Sta=5084,5088
Exp/Cntr=0.3,0.1

Type RM Length L Ch R = 1,56509,232,232,232
BEGIN DESCRIPTION:
Morris Branch 103.0
END DESCRIPTION:
XS GIS Cut Line= 3
      2285778.99      7125259.97      2285679.00      7125010.00
      2285379.00      7124710.00
#Sta/Elev= 30
  4730.5  915.14  4762.8  914.53  4793.7  911.27  4828.8  910.23  4877.2  908.04
  4882.6  908.23  4892.0  907.67  4931.1  906.43  4945.9  906.24  4955.3  905.75
  4960.7  906.37  4967.4  905.89  4978.2  906.02  4997.0  905.07  5013.9  905.01
  5026.0  903.22  5026.3  902.72  5029.8  902.72  5030.0  903.22  5042.2  905.23
  5056.3  905.53  5098.7  904.64  5141.2  905.76  5155.3  906.43  5183.6  906.72
  5254.3  908.76  5296.7  910.84  5409.9  915.44  5420.5  916.36  5424.0  916.36
#Mann=3,-1,0
  4730.5    0.05       0  5026.0   0.033       0  5030.0    0.05       0
Bank Sta=5026,5030
Exp/Cntr=0.3,0.1

Type RM Length L Ch R = 1,56277,72,72,72
BEGIN DESCRIPTION:
Mapping XS c3412025
END DESCRIPTION:
XS GIS Cut Line= 4
      2285903.26      7125123.13      2285888.98      7124910.90
      2285870.17      7124789.51      2285755.65      7124595.77
#Sta/Elev= 30
  4836.7  910.51  4869.9  909.09  4910.0  906.59  4969.9  904.39  5010.2  903.96
  5020.2  904.39  5040.3  904.26  5052.4  903.91  5070.6  902.83  5078.8  901.99
  5083.8  902.51  5090.8  901.67  5178.9  901.19  5179.2  900.69  5182.7  900.69
  5182.9  901.19  5245.3  901.67  5253.0  902.39  5260.9  903.59  5266.7  903.79
  5276.2  905.16  5298.0  904.90  5325.2  905.63  5346.7  906.78  5362.3  908.00
  5369.2  907.90  5377.9  907.03  5383.7  907.31  5392.0  908.32  5397.3  908.32
#Mann=3,-1,0
  4836.7    0.05       0  5178.9   0.033       0  5182.9    0.05       0
Bank Sta=5178.9,5182.9
Exp/Cntr=0.3,0.1

Type RM Length L Ch R = 1,56205,332,332,332
BEGIN DESCRIPTION:
Mapping XS 0a1d675c
END DESCRIPTION:
XS GIS Cut Line= 4
      2285961.73      7125097.75      2285965.48      7124903.00
      2285972.11      7124784.02      2285894.61      7124534.63
#Sta/Elev= 30
  4861.4  910.95  4909.2  907.54  4976.8  904.55  4989.2  904.35  4999.2  903.67
  5009.2  902.08  5019.2  901.01  5047.2  899.91  5047.4  899.41  5050.9  899.41
  5051.2  899.91  5055.2  900.28  5069.2  900.04  5079.2  901.37  5089.2  900.89
  5099.2  902.19  5109.3  902.36  5159.3  902.00  5180.1  902.17  5190.0  900.95
  5211.0  901.43  5231.5  902.38  5236.8  901.35  5242.4  902.40  5263.3  902.87
  5269.3  902.62  5274.6  902.96  5284.3  902.63  5367.0  904.96  5436.5  905.75
#Mann=3,-1,0
  4861.4    0.05       0  5047.2   0.033       0  5051.2    0.05       0
#XS Ineff=2,0
       0                 5127.30    0.00  905.87
Permanent Ineff=
       F       F
Bank Sta=5047.2,5051.2
Exp/Cntr=0.3,0.1

Type RM Length L Ch R = 1,55873,210,210,210
BEGIN DESCRIPTION:
Mapping XS 6236102f
END DESCRIPTION:
XS GIS Cut Line= 2
      2286299.27      7124999.33      2286031.00      7124531.37
#Sta/Elev= 30
  4699.7  909.66  4707.5  909.00  4713.3  909.33  4729.1  908.08  4734.8  908.27
  4744.9  907.53  4750.7  907.60  4788.0  905.21  4793.8  905.38  4809.6  904.41
  4831.2  904.05  4847.0  903.12  4874.4  902.42  4883.4  901.72  4911.8  901.23
  4917.9  900.50  4941.0  900.02  4976.5  900.12  4992.3  898.56  4998.6  898.63
  5011.9  897.75  5012.2  897.25  5015.7  897.25  5015.9  897.75  5021.7  900.12
  5029.7  900.84  5079.3  900.87  5102.4  901.63  5190.8  902.84  5239.1  904.05
#Mann=3,-1,0
  4699.7    0.05       0  5011.9   0.033       0  5015.9    0.05       0
#XS Ineff=2,0
    0.00 4959.30  904.94               0
Permanent Ineff=
       F       F
Bank Sta=5011.9,5015.9
Exp/Cntr=0.3,0.1

Type RM Length L Ch R = 1,55663,354,354,354
BEGIN DESCRIPTION:
Morris Branch 100.0
END DESCRIPTION:
XS GIS Cut Line= 3
      2286479.00      7124910.00      2286279.00      7124610.00
      2285979.01      7124410.00
#Sta/Elev= 30
  4640.2  910.03  4647.7  909.50  4653.7  910.43  4662.7  910.01  4668.7  908.91
  4740.9  905.77  4791.9  902.83  4820.5  902.12  4828.0  901.49  4885.1  899.66
  4900.1  898.07  4921.1  898.17  4928.6  896.29  4936.2  895.65  4964.7  895.44
  4970.2  894.78  4970.5  894.28  4974.0  894.28  4974.2  894.78  4978.2  895.63
  4987.2  895.35  4993.2  896.24  5003.8  896.22  5008.3  895.59  5029.3  897.56
  5044.3  898.00  5065.4  897.39  5072.9  898.19  5108.9  899.68  5361.3  906.80
#Mann=3,-1,0
  4640.2    0.05       0  4970.2   0.033       0  4974.2    0.05       0
Bank Sta=4970.2,4974.2
Exp/Cntr=0.3,0.1

Type RM Length L Ch R = 1,55309,369,369,369
BEGIN DESCRIPTION:
Morris Branch 99.0
END DESCRIPTION:
XS GIS Cut Line= 3
      2286579.00      7124659.99      2286479.00      7124360.00
      2286428.99      7124159.98
#Sta/Elev= 30
  4688.7  901.70  4794.1  898.94  4899.5  897.37  4920.6  896.80  4941.7  896.66
  4962.8  897.03  4973.3  894.79  4983.8  893.85  4992.4  890.72  4992.6  890.22
  4996.1  890.22  4996.4  890.72  5002.3  891.44  5007.5  891.44  5015.2  895.05
  5064.2  893.95  5069.3  893.48  5077.1  893.28  5097.7  893.00  5105.4  893.04
  5110.6  894.26  5118.3  894.41  5128.6  894.50  5146.7  893.69  5151.8  894.33
  5159.5  896.99  5169.8  899.64  5180.2  900.76  5187.9  901.25  5211.1  902.02
#Mann=3,-1,0
  4688.7    0.05       0  4992.4   0.033       0  4996.4    0.05       0
Bank Sta=4992.4,4996.4
Exp/Cntr=0.3,0.1

Type RM Length L Ch R = 1,54940,200,200,200
BEGIN DESCRIPTION:
Mapping XS 86284ec3
END DESCRIPTION:
XS GIS Cut Line= 2
      2286768.60      7124458.58      2286654.98      7124023.68
#Sta/Elev= 30
  4692.0  897.27  4773.2  894.79  4783.6  894.93  4789.0  894.77  4794.2  895.11
  4845.6  894.56  4855.9  894.20  4876.6  893.98  4905.2  893.35  4910.4  893.39
  4928.3  892.77  4945.7  891.89  4979.9  891.62  4991.3  892.08  5000.6  890.67
  5008.9  886.69  5009.2  886.19  5012.7  886.19  5012.9  886.69  5021.3  889.14
  5026.6  892.40  5031.7  892.99  5052.3  893.72  5061.9  894.38  5067.0  895.50
  5073.0  897.56  5093.6  897.87  5114.3  898.70  5135.0  899.03  5141.5  898.88
#Mann=3,-1,0
  4692.0    0.05       0  5008.9   0.033       0  5012.9    0.05       0
Bank Sta=5008.9,5012.9
Exp/Cntr=0.3,0.1

Type RM Length L Ch R = 1,54740,286,286,286
BEGIN DESCRIPTION:
Mapping XS 270ef40c
END DESCRIPTION:
XS GIS Cut Line= 2
      2286958.34      7124406.38      2286767.15      7123894.31
#Sta/Elev= 30
  4591.2  896.71  4598.0  896.38  4608.8  895.45  4628.5  895.26  4633.8  895.92
  4651.4  895.82  4683.4  894.98  4719.4  894.53  4758.1  893.68  4811.5  892.16
  4885.2  891.24  4890.5  891.35  4896.9  891.00  4945.8  890.13  4993.0  890.29
  5001.1  889.50  5004.4  888.55  5004.7  888.05  5008.2  888.05  5008.4  888.55
  5014.3  888.69  5031.4  890.28  5036.7  892.63  5046.3  892.53  5061.7  893.68
  5086.7  894.44  5092.0  894.81  5117.0  895.10  5122.3  895.36  5137.8  895.37
#Mann=3,-1,0
  4591.2    0.05       0  5004.4   0.033       0  5008.4    0.05       0
Bank Sta=5004.4,5008.4
Exp/Cntr=0.3,0.1

Type RM Length L Ch R = 1,54454,324,324,324
BEGIN DESCRIPTION:
Mapping XS 2be9a3f9
END DESCRIPTION:
XS GIS Cut Line= 3
      2287147.74      7124204.79      2287033.37      7123811.90
      2286792.60      7123824.58
#Sta/Elev= 30
  4692.6  893.17  4737.9  891.94  4743.1  891.42  4776.6  890.93  4781.8  890.03
  4810.1  888.91  4848.8  889.10  4854.1  889.76  4887.6  889.79  4947.5  888.01
  4988.1  887.93  4993.3  888.24  5010.0  885.93  5020.5  885.99  5024.8  884.10
  5025.1  883.60  5028.6  883.60  5028.8  884.10  5032.0  885.74  5041.3  887.76
  5060.3  887.66  5072.5  888.07  5099.1  887.80  5126.2  888.22  5136.2  888.75
  5196.3  890.18  5256.4  890.99  5316.5  893.19  5336.5  893.38  5342.9  893.85
#Mann=3,-1,0
  4692.6    0.05       0  5024.8   0.033       0  5028.8    0.05       0
Bank Sta=5024.8,5028.8
Exp/Cntr=0.3,0.1

Type RM Length L Ch R = 1,54130,296,296,296
BEGIN DESCRIPTION:
Mapping XS 85c1d1dc
END DESCRIPTION:
XS GIS Cut Line= 3
      2287395.11      7124050.69      2287283.69      7123625.28
      2287204.26      7123464.49
#Sta/Elev= 30
  4648.0  894.60  4679.7  893.17  4688.4  892.44  4693.5  892.58  4728.8  889.67
  4733.9  889.71  4783.1  887.44  4885.2  885.04  4938.2  884.69  4948.5  884.82
  4958.8  885.64  4987.8  883.94  4988.1  883.44  4991.6  883.44  4991.8  883.94
  5000.2  884.28  5011.6  886.09  5041.5  885.22  5052.0  885.73  5082.1  885.56
  5087.1  886.01  5104.4  886.01  5110.0  886.46  5126.9  886.36  5160.6  887.20
  5194.0  887.22  5205.4  887.72  5244.7  888.19  5250.2  888.67  5267.1  888.84
#Mann=3,-1,0
  4648.0    0.05       0  4987.8   0.033       0  4991.8    0.05       0
Bank Sta=4987.8,4991.8
Exp/Cntr=0.3,0.1

Type RM Length L Ch R = 1,53834,446,446,446
BEGIN DESCRIPTION:
Mapping XS dcabce46
END DESCRIPTION:
XS GIS Cut Line= 2
      2287694.20      7123782.39      2287323.64      7123248.36
#Sta/Elev= 30
  4757.5  891.66  4762.2  890.77  4770.9  890.64  4777.0  889.89  4798.0  888.93
  4806.7  888.83  4812.8  888.09  4827.7  888.31  4857.4  887.26  4870.0  886.55
  4893.2  884.24  4899.3  883.97  4920.2  884.05  4935.1  883.55  4943.0  884.26
  4956.0  883.38  4985.7  883.73  5000.6  882.83  5028.2  883.23  5057.3  882.59
  5062.7  882.16  5062.9  881.66  5066.4  881.66  5066.7  882.16  5072.2  882.70
  5093.1  882.59  5108.0  883.29  5149.9  884.22  5316.7  886.25  5407.5  888.00
#Mann=3,-1,0
  4757.5    0.05       0  5062.7   0.033       0  5066.7    0.05       0
Bank Sta=5062.7,5066.7
Exp/Cntr=0.3,0.1

Type RM Length L Ch R = 1,53388,413,413,413
BEGIN DESCRIPTION:
Mapping XS 104d0155
END DESCRIPTION:
XS GIS Cut Line= 3
      2287998.24      7123516.15      2287669.16      7123026.50
      2287433.53      7123026.09
#Sta/Elev= 30
  4657.0  895.61  4697.5  894.93  4712.5  893.74  4718.5  892.46  4739.5  890.10
  4769.5  888.04  4775.5  886.80  4796.9  886.09  4805.5  884.47  4841.5  880.96
  4856.5  880.30  4883.5  881.22  4898.5  880.55  4911.5  877.13  4911.8  876.63
  4915.3  876.63  4915.5  877.13  4928.5  880.39  4941.5  881.45  4970.5  881.33
  4977.7  880.57  4985.5  878.46  4991.5  880.31  5000.5  881.52  5006.5  881.10
  5021.5  881.74  5042.5  880.21  5063.5  881.33  5249.5  882.60  5482.6  887.40
#Mann=3,-1,0
  4657.0    0.05       0  4911.5   0.033       0  4915.5    0.05       0
Bank Sta=4911.5,4915.5
Exp/Cntr=0.3,0.1

Type RM Length L Ch R = 1,52975,357,357,357
BEGIN DESCRIPTION:
Mapping XS 85784e65
END DESCRIPTION:
XS GIS Cut Line= 2
      2288221.58      7123211.67      2287675.01      7122551.72
#Sta/Elev= 30
  4648.9  886.32  4829.8  879.85  4865.0  879.80  4893.6  879.04  4907.9  878.01
  4943.1  877.88  4986.1  876.92  4992.6  875.66  5000.4  875.02  5004.8  873.33
  5005.1  872.83  5008.7  872.83  5009.1  873.33  5021.2  874.51  5027.7  878.72
  5120.2  879.45  5148.9  880.53  5184.0  880.93  5191.9  880.45  5198.4  880.83
  5212.7  880.01  5227.0  880.89  5255.7  880.65  5262.2  881.73  5270.0  881.85
  5290.8  883.52  5333.8  884.71  5376.8  886.65  5412.0  887.19  5505.8  890.90
#Mann=3,-1,0
  4648.9    0.05       0  5004.8   0.033       0  5009.1    0.05       0
Bank Sta=5004.8,5009.1
Exp/Cntr=0.3,0.1

Type RM Length L Ch R = 1,52618,400,400,400
BEGIN DESCRIPTION:
Mapping XS 287a74bc
END DESCRIPTION:
XS GIS Cut Line= 4
      2288384.31      7122950.11      2288069.31      7122424.06
      2288066.39      7122424.03      2287874.85      7122366.73
#Sta/Elev= 30
  4713.1  882.32  4864.2  878.44  4885.6  877.31  4899.7  877.02  4907.0  878.02
  4912.8  877.93  4934.7  876.25  4958.0  875.42  4980.8  875.20  4986.7  874.62
  4993.0  871.81  5000.1  871.37  5000.4  870.87  5004.0  870.87  5004.4  871.37
  5008.1  874.95  5016.3  875.68  5039.2  874.89  5097.5  874.71  5124.7  875.06
  5140.3  874.60  5214.2  874.46  5262.8  877.16  5299.8  878.19  5336.9  878.45
  5378.6  880.69  5466.4  883.34  5472.6  884.12  5499.5  885.95  5529.1  887.01
#Mann=3,-1,0
  4713.1    0.05       0  5000.1   0.033       0  5004.4    0.05       0
Bank Sta=5000.1,5004.4
Exp/Cntr=0.3,0.1

Type RM Length L Ch R = 1,52218,225,225,225
BEGIN DESCRIPTION:
Mapping XS b8865ab3
END DESCRIPTION:
XS GIS Cut Line= 3
      2288665.55      7122746.19      2288347.27      7122254.71
      2287772.64      7122212.72
#Sta/Elev= 30
  4585.7  881.15  4608.9  880.27  4616.9  881.08  4624.1  879.31  4652.6  878.48
  4660.4  877.62  4883.9  873.73  4896.9  872.76  4897.3  872.26  4900.9  872.26
  4901.2  872.76  4926.7  874.32  4956.5  874.52  4971.6  873.63  4986.2  873.72
  4998.7  875.05  5007.9  874.64  5013.8  873.35  5044.2  874.45  5050.1  873.50
  5071.2  873.14  5189.6  873.78  5400.1  877.21  5550.5  882.90  5577.2  885.11
  5582.2  884.55  5620.7  887.56  5680.9  889.70  5731.0  890.71  5747.4  890.25
#Mann=3,-1,0
  4585.7    0.05       0  4896.9   0.033       0  4901.2    0.05       0
Bank Sta=4896.9,4901.2
Exp/Cntr=0.3,0.1

Type RM Length L Ch R = 1,51993,765,765,765
BEGIN DESCRIPTION:
Mapping XS 24bc437b
END DESCRIPTION:
XS GIS Cut Line= 4
      2288692.97      7122621.72      2288695.56      7122362.07
      2288410.63      7122031.97      2288062.49      7122064.71
#Sta/Elev= 30
  4563.1  878.24  4634.8  877.34  4668.1  877.46  4704.8  876.67  4714.8  875.99
  4724.8  876.16  4850.5  873.55  4885.7  871.26  4892.3  870.15  4897.7  869.90
  4898.1  869.40  4901.7  869.40  4902.1  869.90  4906.5  870.87  4920.8  871.35
  4928.4  872.54  4942.7  872.66  4956.9  871.69  4984.4  871.73  4992.1  871.36
  4998.7  870.17  5012.9  871.64  5027.2  871.92  5070.0  870.83  5105.1  872.22
  5155.5  871.71  5262.2  873.04  5461.3  877.05  5471.4  877.59  5608.5  879.67
#Mann=3,-1,0
  4563.1    0.05       0  4897.7   0.033       0  4902.1    0.05       0
Bank Sta=4897.7,4902.1
Exp/Cntr=0.3,0.1

Type RM Length L Ch R = 1,51228,308,308,308
BEGIN DESCRIPTION:
Mapping XS 7fbf783b
END DESCRIPTION:
XS GIS Cut Line= 2
      2289163.98      7122130.24      2288484.01      7121420.50
#Sta/Elev= 30
  4536.6  883.94  4575.7  882.32  4632.4  878.15  4653.4  875.72  4717.0  871.97
  4809.1  870.16  4851.6  870.21  4858.5  869.43  4865.7  867.51  4879.9  865.05
  4894.0  865.58  4900.9  865.03  4908.2  865.99  4922.3  866.42  4957.5  865.55
  4978.9  866.09  5000.0  865.89  5007.2  864.68  5011.6  862.11  5012.3  861.61
  5016.1  861.61  5016.8  862.11  5021.4  864.45  5028.3  865.76  5141.5  869.92
  5226.4  874.67  5233.4  875.56  5254.7  875.93  5445.6  883.19  5519.5  887.19
#Mann=3,-1,0
  4536.6    0.05       0  5011.6   0.033       0  5016.8    0.05       0
Bank Sta=5011.6,5016.8
Exp/Cntr=0.3,0.1

Type RM Length L Ch R = 1,50920,403,403,403
BEGIN DESCRIPTION:
Morris Branch 88.0
END DESCRIPTION:
XS GIS Cut Line= 3
      2289279.02      7121960.03      2289029.00      7121560.00
      2288629.01      7121160.01
#Sta/Elev= 30
  4524.1  884.17  4568.4  882.98  4583.1  879.86  4589.6  877.11  4604.9  874.08
  4618.5  874.31  4668.6  870.91  4748.2  867.75  4799.5  867.57  4909.2  865.24
  4915.1  865.72  4960.5  865.37  4972.8  864.31  4982.3  864.25  4988.2  863.31
  4999.4  863.65  5007.4  861.24  5008.1  860.74  5011.9  860.74  5012.6  861.24
  5024.1  862.89  5038.3  863.81  5066.5  862.45  5109.0  868.94  5137.3  870.77
  5222.1  873.05  5391.8  880.40  5406.0  881.81  5476.7  885.27  5561.5  891.06
#Mann=3,-1,0
  4524.1    0.05       0  5007.4   0.033       0  5012.6    0.05       0
Bank Sta=5007.4,5012.6
Exp/Cntr=0.3,0.1

Type RM Length L Ch R = 1,50517,443,443,443
BEGIN DESCRIPTION:
Morris Branch 87.0
END DESCRIPTION:
XS GIS Cut Line= 3
      2289329.00      7121960.01      2289179.00      7121260.00
      2288779.01      7120910.01
#Sta/Elev= 30
  4292.1  883.78  4343.2  881.90  4435.3  872.92  4476.2  870.64  4568.2  867.44
  4721.6  864.83  4752.3  861.69  4823.9  861.33  4840.1  859.22  4845.2  860.57
  4884.4  858.85  4889.5  860.57  4895.5  860.92  4926.2  860.24  4939.0  862.13
  4983.3  861.96  4988.4  863.05  5005.4  860.97  5021.8  860.14  5026.8  857.88
  5027.5  857.38  5032.0  857.88  5036.0  860.33  5057.8  860.57  5072.1  862.89
  5086.3  867.18  5114.3  869.78  5305.6  877.85  5426.1  884.70  5539.5  893.01
#Mann=3,-1,0
  4292.1    0.05       0  5026.8   0.033       0  5032.0    0.05       0
Bank Sta=5026.8,5032
Exp/Cntr=0.3,0.1

Type RM Length L Ch R = 1,50074,453,453,453
BEGIN DESCRIPTION:
Morris Branch 86.0
END DESCRIPTION:
XS GIS Cut Line= 3
      2289879.00      7121510.00      2289479.00      7121110.00
      2289078.98      7120709.98
#Sta/Elev= 30
  4429.7  878.51  4500.4  873.01  4557.0  866.90  4585.3  865.46  4627.7  863.91
  4641.8  864.37  4670.1  864.05  4684.3  863.11  4740.8  863.37  4811.5  862.08
  4967.1  861.45  4981.2  860.72  4991.9  859.33  4998.9  859.33  5006.9  857.04
  5007.6  856.54  5011.4  856.54  5012.2  857.04  5023.7  859.41  5052.0  859.64
  5066.1  859.04  5108.5  861.26  5122.7  861.26  5136.8  861.90  5165.1  864.96
  5235.8  866.81  5264.1  868.26  5292.4  870.56  5476.2  879.36  5561.1  884.52
#Mann=3,-1,0
  4429.7    0.05       0  5006.9   0.033       0  5012.2    0.05       0
Bank Sta=5006.9,5012.2
Exp/Cntr=0.3,0.1

Type RM Length L Ch R = 1,49621,495,495,495
BEGIN DESCRIPTION:
Morris Branch 85.0
END DESCRIPTION:
XS GIS Cut Line= 3
      2289979.01      7121510.04      2289679.00      7120760.00
      2289478.97      7120709.99
#Sta/Elev= 30
  4195.5  881.55  4258.8  878.50  4281.7  873.87  4288.4  870.74  4293.8  869.48
  4324.8  867.39  4420.4  866.55  4509.2  866.78  4533.5  866.05  4540.2  862.14
  4551.0  860.89  4587.3  860.97  4611.5  860.20  4778.5  858.32  4827.0  858.84
  4841.8  857.99  4934.7  856.74  4964.3  857.48  4971.0  856.84  4988.5  856.84
  4993.9  856.35  4997.8  855.07  4998.7  854.57  5003.4  855.07  5005.9  855.07
  5013.6  857.51  5021.4  860.82  5044.5  866.25  5096.1  866.52  5209.5  870.09
#Mann=3,-1,0
  4195.5    0.05       0  4997.8   0.033       0  5003.4    0.05       0
Bank Sta=4997.8,5003.4
Exp/Cntr=0.3,0.1

Type RM Length L Ch R = 1,49126,361,361,361
BEGIN DESCRIPTION:
Mapping XS e75557ba
END DESCRIPTION:
XS GIS Cut Line= 3
      2290131.09      7121201.43      2290009.02      7120597.63
      2289815.71      7120426.04
#Sta/Elev= 30
  4651.2  869.26  4662.9  869.94  4693.5  863.37  4713.9  861.31  4789.1  858.93
  4805.7  857.54  4815.9  855.82  4866.9  855.33  4885.5  854.43  4917.9  855.89
  4941.4  855.91  4958.7  854.65  4987.0  853.80  4992.1  854.39  4996.7  851.29
  4997.6  850.79  5001.5  850.79  5002.3  851.29  5009.7  852.18  5019.9  855.48
  5030.1  857.64  5071.0  858.28  5081.2  857.54  5190.0  857.74  5286.8  860.54
  5364.5  861.08  5435.6  862.96  5442.3  863.63  5478.3  864.78  5525.7  865.03
#Mann=3,-1,0
  4651.2    0.05       0  4996.7   0.033       0  5002.3    0.05       0
Bank Sta=4996.7,5002.3
Exp/Cntr=0.3,0.1

Type RM Length L Ch R = 1,48765,473,473,473
BEGIN DESCRIPTION:
Mapping XS 53d91fe5
END DESCRIPTION:
XS GIS Cut Line= 3
      2290411.66      7121093.43      2290325.82      7120652.74
      2290053.17      7120346.23
#Sta/Elev= 30
  4857.2  873.84  4881.1  873.24  4911.6  871.55  4948.4  862.06  4972.8  859.82
  5000.1  858.17  5005.2  856.84  5013.5  851.31  5020.9  848.85  5021.8  848.35
  5025.7  848.35  5026.5  848.85  5044.1  851.62  5056.8  852.82  5074.6  853.50
  5095.0  853.62  5125.6  853.04  5135.8  853.98  5176.5  855.25  5196.9  854.57
  5211.6  854.43  5217.3  855.01  5227.5  854.25  5258.0  854.06  5341.2  854.72
  5348.7  854.32  5510.9  856.30  5567.8  858.07  5659.7  860.13  5716.4  860.40
#Mann=3,-1,0
  4857.2    0.05       0  5020.9   0.033       0  5026.5    0.05       0
Bank Sta=5020.9,5026.5
Exp/Cntr=0.3,0.1

Type RM Length L Ch R = 1,48292,469,469,469
BEGIN DESCRIPTION:
Morris Branch 82.0
END DESCRIPTION:
XS GIS Cut Line= 4
      2290979.00      7120810.00      2290579.00      7120560.00
      2290409.17      7120333.56      2290087.63      7120345.05
#Sta/Elev= 30
  4528.9  866.35  4630.9  862.24  4658.6  861.47  4667.5  861.71  4776.5  858.31
  4840.8  855.77  4862.0  855.56  4941.6  852.25  4956.4  852.09  4965.2  850.06
  4971.7  846.75  4974.7  846.16  4975.6  845.66  4979.6  845.66  4980.6  846.16
  4987.0  848.16  4992.9  848.96  4997.7  850.52  5014.1  851.11  5078.7  851.14
  5093.3  850.15  5122.5  851.06  5157.9  853.13  5200.6  854.35  5264.1  855.40
  5286.2  855.07  5363.9  856.94  5403.9  856.92  5453.9  858.29  5605.4  859.94
#Mann=3,-1,0
  4528.9    0.05       0  4974.7   0.033       0  4980.6    0.05       0
Bank Sta=4974.7,4980.6
Exp/Cntr=0.3,0.1

Type RM Length L Ch R = 1,47823,421,421,421
BEGIN DESCRIPTION:
Morris Branch 81.0
END DESCRIPTION:
XS GIS Cut Line= 3
      2291178.97      7120559.98      2290829.00      7120310.00
      2290328.99      7119509.98
#Sta/Elev= 30
  4570.2  867.10  4734.8  858.68  4951.1  854.45  4978.2  851.68  4986.8  848.40
  4990.0  845.21  4990.9  844.71  4995.9  845.21  4997.2  846.56  5029.2  849.47
  5130.0  849.24  5175.4  847.54  5189.0  848.87  5202.5  847.44  5217.9  848.66
  5224.3  850.26  5233.2  849.32  5239.1  850.80  5254.4  849.33  5291.0  848.85
  5333.4  850.72  5354.6  853.15  5479.6  855.64  5589.3  859.56  5660.7  866.11
  5719.6  868.77  5762.7  872.77  5841.7  877.10  5857.0  879.33  5943.7  885.48
#Mann=3,-1,0
  4570.2    0.05       0  4990.0    0.04       0  4995.9    0.05       0
Bank Sta=4990,4995.9
Exp/Cntr=0.3,0.1

Type RM Length L Ch R = 1,47402,424,424,424
BEGIN DESCRIPTION:
Morris Branch 80.0
END DESCRIPTION:
XS GIS Cut Line= 3
      2291178.99      7120409.99      2290879.00      7120010.00
      2290478.98      7119609.98
#Sta/Elev= 30
  4500.3  861.89  4513.8  860.34  4572.2  857.44  4593.0  857.26  4622.2  855.04
  4700.3  852.74  4743.0  852.41  4807.6  850.66  4836.7  850.61  4843.0  851.49
  4857.6  851.23  4878.4  849.92  4907.6  849.44  4957.6  849.67  4963.8  847.02
  4983.4  844.94  4984.5  844.44  4989.0  844.44  4990.0  844.94  4993.0  845.49
  5003.8  844.96  5014.4  846.70  5028.6  846.15  5056.9  846.37  5113.4  848.35
  5212.4  853.22  5325.6  857.36  5495.3  868.34  5537.7  872.87  5566.0  874.90
#Mann=3,-1,0
  4500.3    0.05       0  4983.4    0.04       0  4990.0    0.05       0
Bank Sta=4983.4,4990
Exp/Cntr=0.3,0.1

Type RM Length L Ch R = 1,46978,534,534,534
BEGIN DESCRIPTION:
Morris Branch 79.0
END DESCRIPTION:
XS GIS Cut Line= 3
      2291279.01      7120410.03      2290979.00      7119660.00
      2290879.00      7119610.00
#Sta/Elev= 30
  4191.9  864.98  4224.2  864.45  4255.2  862.24  4260.6  861.70  4267.3  860.30
  4284.8  858.76  4338.7  855.24  4428.9  851.62  4476.0  850.51  4524.5  848.31
  4686.0  846.96  4784.3  847.28  4853.0  846.36  4882.6  847.51  4913.5  845.44
  4955.3  845.90  4960.7  845.20  4984.9  844.90  4990.3  842.97  4993.7  842.38
  4994.8  841.88  4999.3  841.88  5000.3  842.38  5008.1  842.46  5013.7  843.23
  5030.4  849.73  5052.8  852.17  5075.2  853.80  5080.8  855.18  5111.5  857.43
#Mann=3,-1,0
  4191.9    0.05       0  4993.7   0.033       0  5000.3    0.05       0
Bank Sta=4993.7,5000.3
Exp/Cntr=0.3,0.1

Type RM Length L Ch R = 1,46444,773,773,773
BEGIN DESCRIPTION:
Mapping XS cb2ee72a
END DESCRIPTION:
XS GIS Cut Line= 2
      2291513.37      7120176.34      2291239.21      7119234.21
#Sta/Elev= 30
  4151.8  852.38  4218.4  848.66  4257.1  847.52  4314.6  845.19  4368.1  844.26
  4460.4  843.51  4540.9  843.52  4606.2  844.30  4646.6  843.43  4679.1  843.24
  4710.4  844.39  4718.9  845.17  4731.2  844.69  4791.1  845.15  4814.5  844.97
  4829.9  844.42  4902.1  844.57  5002.0  843.55  5013.1  842.11  5019.5  840.72
  5020.6  840.22  5025.1  840.22  5026.2  840.72  5033.2  842.90  5041.4  848.34
  5054.1  856.02  5085.3  858.96  5106.1  859.79  5118.8  861.20  5133.0  862.12
#Mann=3,-1,0
  4151.8    0.05       0  5019.5    0.04       0  5026.2    0.05       0
#XS Ineff=2,0
    0.00 4748.00  851.50               0
Permanent Ineff=
       F       F
Bank Sta=5019.5,5026.2
Exp/Cntr=0.3,0.1

Type RM Length L Ch R = 1,45671,375,375,375
BEGIN DESCRIPTION:
Mapping XS 04ceeaa8
END DESCRIPTION:
XS GIS Cut Line= 2
      2291816.15      7120034.01      2291791.67      7118994.90
#Sta/Elev= 30
  4676.1  847.52  4860.2  843.41  4930.2  842.85  4940.2  843.71  4960.2  841.94
  4966.7  837.09  4967.8  836.59  4972.5  836.59  4973.6  837.09  4980.2  839.21
  4990.2  838.11  5000.2  839.57  5010.2  839.95  5120.2  841.51  5160.2  841.06
  5260.3  841.56  5340.3  843.26  5370.3  844.57  5380.3  844.26  5390.3  845.09
  5400.3  844.91  5450.3  846.35  5490.3  848.28  5540.4  849.23  5560.4  851.39
  5580.4  851.09  5630.4  853.87  5650.4  853.94  5710.4  858.66  5715.5  859.56
#Mann=3,-1,0
  4676.1    0.05       0  4966.7   0.033       0  4973.6    0.05       0
Bank Sta=4966.7,4973.6
Exp/Cntr=0.3,0.1

Type RM Length L Ch R = 1,45296,614,614,614
BEGIN DESCRIPTION:
Mapping XS 8bea98e1
END DESCRIPTION:
XS GIS Cut Line= 2
      2292170.83      7119941.45      2291979.65      7118975.89
#Sta/Elev= 30
  4596.6  845.78  4730.1  841.60  4802.0  840.74  4832.5  839.27  4842.8  840.48
  4852.9  840.50  4883.5  838.86  5005.8  838.20  5016.0  836.42  5022.7  833.49
  5023.8  832.99  5029.8  833.49  5042.6  838.58  5056.8  839.20  5145.0  839.42
  5219.9  840.94  5230.1  841.90  5252.6  840.39  5311.7  843.66  5342.2  844.15
  5349.9  843.66  5372.8  844.96  5406.3  845.16  5413.6  846.15  5423.8  845.96
  5474.8  848.29  5485.0  847.93  5554.9  852.59  5566.5  855.47  5580.9  856.62
#Mann=3,-1,0
  4596.6    0.05       0  5022.7    0.04       0  5029.8    0.05       0
Bank Sta=5022.7,5029.8
Exp/Cntr=0.3,0.1

Type RM Length L Ch R = 1,44682,454,454,454
BEGIN DESCRIPTION:
Morris Branch 74.0
END DESCRIPTION:
XS GIS Cut Line= 3
      2292528.99      7120009.98      2292279.00      7119260.00
      2292029.02      7118860.04
#Sta/Elev= 30
  4213.1  848.89  4286.9  847.34  4392.3  843.15  4423.9  843.87  4582.0  838.75
  4676.9  838.11  4687.4  835.71  4708.5  834.06  4792.8  835.68  4803.4  834.67
  4813.9  836.61  4908.8  836.69  4961.5  835.86  4997.4  833.79  4998.6  833.29
  5004.6  833.79  5011.3  833.90  5032.5  838.40  5062.6  838.29  5126.9  842.64
  5133.4  841.40  5169.3  841.77  5192.3  843.79  5200.0  842.20  5236.5  845.39
  5263.7  845.17  5345.6  849.62  5388.7  856.47  5440.0  860.23  5475.3  864.72
#Mann=3,-1,0
  4213.1    0.05       0  4997.4   0.033       0  5004.6    0.05       0
Bank Sta=4997.4,5004.6
Exp/Cntr=0.3,0.1

Type RM Length L Ch R = 1,44228,469,469,469
BEGIN DESCRIPTION:
Morris Branch 73.0
END DESCRIPTION:
XS GIS Cut Line= 3
      2292778.99      7119659.97      2292679.00      7119260.00
      2292278.98      7118859.98
#Sta/Elev= 30
  4591.8  845.56  4715.5  842.61  4738.7  841.62  4787.6  838.07  4808.2  837.51
  4828.8  835.50  4857.2  834.58  4962.8  834.50  4973.2  833.47  4980.9  831.61
  4986.0  829.50  4990.2  829.24  4991.3  828.74  4997.4  829.24  5001.5  830.08
  5007.6  830.08  5018.2  832.71  5074.8  832.79  5117.2  834.88  5216.2  835.95
  5286.9  839.63  5329.3  839.25  5428.3  842.82  5456.6  842.76  5484.9  845.29
  5499.1  844.97  5527.3  848.90  5541.5  849.91  5566.2  853.61  5569.8  853.61
#Mann=3,-1,0
  4591.8    0.05       0  4990.2   0.033       0  4997.4    0.05       0
Bank Sta=4990.2,4997.4
Exp/Cntr=0.3,0.1

Type RM Length L Ch R = 1,43759,567,567,567
BEGIN DESCRIPTION:
Morris Branch 72.0
END DESCRIPTION:
XS GIS Cut Line= 3
      2292879.00      7119659.97      2292929.00      7119010.00
      2292779.02      7118760.03
#Sta/Elev= 30
  4348.0  846.20  4378.1  844.75  4468.3  843.84  4528.5  842.13  4578.6  836.83
  4638.8  834.08  4719.1  833.51  4769.2  832.49  4889.6  833.64  4899.6  833.46
  4929.7  830.94  4969.8  831.54  5002.8  829.10  5007.7  826.20  5019.6  825.48
  5020.7  824.98  5025.7  824.98  5026.9  825.48  5034.9  826.68  5044.6  832.08
  5050.4  833.40  5058.2  834.02  5174.8  834.35  5225.4  837.52  5233.1  838.91
  5240.9  841.63  5246.7  842.63  5256.4  846.15  5268.1  848.92  5291.4  852.09
#Mann=3,-1,0
  4348.0    0.05       0  5019.6    0.04       0  5026.9    0.05       0
Bank Sta=5019.6,5026.9
Exp/Cntr=0.3,0.1

Type RM Length L Ch R = 1,43192,294,294,294
BEGIN DESCRIPTION:
Morris Branch 71.0
END DESCRIPTION:
XS GIS Cut Line= 3
      2293729.01      7119610.01      2293422.62      7119136.98
      2293371.99      7118103.91
#Sta/Elev= 30
  4158.9  852.34  4217.9  849.38  4239.0  847.03  4368.9  841.16  4426.3  839.69
  4477.7  836.26  4659.1  833.71  4721.2  831.40  4759.5  832.39  4799.6  831.98
  4819.6  829.76  4859.6  827.86  4869.6  828.56  4901.6  828.43  4919.7  827.39
  4939.7  828.83  4959.8  828.17  4989.8  823.20  5015.8  822.38  5017.0  821.88
  5023.9  822.38  5029.8  826.62  5039.8  829.31  5049.9  829.91  5109.9  829.88
  5160.0  828.56  5306.1  830.42  5450.3  832.78  5590.5  836.75  5756.8  839.77
#Mann=3,-1,0
  4158.9    0.05       0  5015.8    0.04       0  5023.9    0.05       0
Bank Sta=5015.8,5023.9
Exp/Cntr=0.3,0.1

Type RM Length L Ch R = 1,42898,440,440,440
BEGIN DESCRIPTION:
Mapping XS 1ef5bedd
END DESCRIPTION:
XS GIS Cut Line= 2
      2293744.96      7119196.20      2293554.88      7118198.65
#Sta/Elev= 30
  4697.4  835.22  4810.0  832.00  4937.9  829.91  4958.2  826.55  4971.6  823.57
  4988.8  822.44  5005.1  822.41  5006.3  821.91  5013.2  822.41  5023.7  822.61
  5029.5  824.45  5039.7  825.19  5049.8  827.06  5075.9  824.81  5081.0  825.46
  5090.6  824.53  5100.7  824.40  5128.0  825.30  5161.8  823.32  5172.0  825.89
  5180.2  828.81  5185.3  829.05  5237.5  828.28  5253.4  829.23  5273.8  827.75
  5314.5  827.37  5426.5  828.30  5518.1  830.00  5619.9  833.21  5712.9  835.32
#Mann=3,-1,0
  4697.4    0.05       0  5005.1   0.033       0  5013.2    0.05       0
Bank Sta=5005.1,5013.2
Exp/Cntr=0.3,0.1

Type RM Length L Ch R = 1,42458,617,617,617
BEGIN DESCRIPTION:
Mapping XS 1281f5b5
END DESCRIPTION:
XS GIS Cut Line= 2
      2294233.59      7119101.55      2293778.14      7118075.38
#Sta/Elev= 30
  4629.9  838.35  4784.8  834.11  4839.5  831.61  4847.8  830.61  4876.6  830.37
  4899.8  829.01  4905.3  829.52  4928.6  828.54  4937.9  827.12  4951.8  823.03
  4969.6  820.72  4977.5  818.72  4978.8  818.22  4985.8  818.72  4992.6  818.90
  4998.4  821.02  5003.8  824.18  5036.4  823.97  5058.3  825.58  5166.7  824.40
  5200.9  825.02  5242.0  826.69  5265.2  826.33  5277.1  827.69  5294.0  826.37
  5317.2  825.98  5375.6  826.52  5444.5  826.17  5560.8  827.46  5752.6  834.06
#Mann=3,-1,0
  4629.9    0.05       0  4977.5   0.033       0  4985.8    0.05       0
Bank Sta=4977.5,4985.8
Exp/Cntr=0.3,0.1

Type RM Length L Ch R = 1,41841,414,414,414
BEGIN DESCRIPTION:
Mapping XS f6f89829
END DESCRIPTION:
XS GIS Cut Line= 2
      2294622.17      7118828.52      2294324.38      7117687.02
#Sta/Elev= 30
  4567.1  843.27  4595.4  843.31  4635.9  839.62  4648.2  834.68  4716.9  817.77
  4772.3  818.67  4803.3  820.74  4833.1  818.79  4838.3  820.47  4854.9  819.22
  4878.8  819.89  4896.3  816.46  4919.3  819.49  4937.6  819.28  4954.6  823.03
  4959.7  820.34  4979.0  822.71  4989.3  822.00  4995.0  819.03  5010.0  818.38
  5025.8  815.56  5027.1  815.06  5035.0  815.56  5035.5  817.04  5041.0  822.18
  5103.0  821.12  5134.0  823.80  5144.3  822.77  5361.3  825.26  5746.8  835.11
#Mann=3,-1,0
  4567.1    0.05       0  5025.8   0.033       0  5035.0    0.05       0
Bank Sta=5025.8,5035
Exp/Cntr=0.3,0.1

Type RM Length L Ch R = 1,41427,579,579,579
BEGIN DESCRIPTION:
Mapping XS 2652aa69
END DESCRIPTION:
XS GIS Cut Line= 2
      2294962.36      7118658.77      2294744.44      7117539.79
#Sta/Elev= 30
  4644.7  836.81  4663.8  836.88  4674.0  835.98  4683.8  834.17  4694.4  827.89
  4704.6  824.25  4714.8  822.32  4740.5  820.30  4765.7  819.75  4816.6  820.80
  4826.8  820.32  4843.7  816.87  4867.6  817.55  4877.8  816.24  4895.4  816.59
  4908.3  818.91  4918.5  819.43  4959.3  818.80  4989.8  820.40  4998.6  819.71
  5010.2  814.28  5015.8  814.06  5017.1  813.56  5025.0  814.06  5030.6  817.03
  5061.1  820.60  5193.6  820.77  5210.2  819.91  5550.2  826.07  5784.7  829.11
#Mann=3,-1,0
  4644.7    0.05       0  5015.8    0.04       0  5025.0    0.05       0
Bank Sta=5015.8,5025
Exp/Cntr=0.3,0.1

Type RM Length L Ch R = 1,40848,1257,1257,1257
BEGIN DESCRIPTION:
Mapping XS 81c959e4
END DESCRIPTION:
XS GIS Cut Line= 2
      2295429.30      7118484.48      2294924.57      7117497.22
#Sta/Elev= 30
  4805.7  825.60  4855.7  824.09  4889.3  821.30  4900.1  821.35  4922.3  820.21
  4950.1  818.06  4956.7  818.39  4966.7  815.45  4967.6  813.31  4969.0  812.81
  4975.7  812.81  4977.0  813.31  4988.9  813.97  4994.6  816.03  5001.7  817.67
  5024.1  818.35  5069.0  817.43  5194.5  817.83  5255.5  816.56  5271.2  816.97
  5344.4  816.53  5361.0  816.83  5366.6  817.71  5383.2  816.90  5494.3  817.00
  5560.9  817.85  5641.8  820.30  5672.0  820.42  5722.0  822.09  5914.5  825.77
#Mann=3,-1,0
  4805.7    0.05       0  4967.6    0.04       0  4977.0    0.05       0
Bank Sta=4967.6,4977
Exp/Cntr=0.3,0.1

Type RM Length L Ch R = 1,39591,791,791,791
BEGIN DESCRIPTION:
Mapping XS 37ab876a
END DESCRIPTION:
XS GIS Cut Line= 3
      2295924.17      7118117.06      2295675.79      7117655.37
      2295157.15      7117402.64
#Sta/Elev= 30
  4089.4  820.64  4150.8  818.49  4222.3  817.45  4260.3  816.01  4276.6  816.34
  4392.7  812.83  4446.2  812.49  4460.8  813.60  4506.2  813.41  4528.1  814.65
  4540.3  813.76  4599.5  814.75  4643.5  814.56  4710.8  812.95  4755.9  812.82
  4772.8  813.85  4795.4  812.47  4817.9  813.21  4868.6  811.90  4885.5  812.62
  4953.2  812.23  4981.3  810.93  4983.5  808.12  4984.9  807.62  4993.1  808.12
  4998.2  810.56  5003.8  811.34  5010.6  815.93  5020.8  817.17  5190.6  822.45
#Mann=3,-1,0
  4089.4    0.05       0  4983.5   0.035       0  4993.1    0.05       0
Bank Sta=4983.5,4993.1
Exp/Cntr=0.3,0.1

Type RM Length L Ch R = 1,38800,375,375,375
BEGIN DESCRIPTION:
Morris Branch 63.0
END DESCRIPTION:
XS GIS Cut Line= 3
      2296128.99      7118309.97      2295829.00      7117110.00
      2295728.99      7116959.98
#Sta/Elev= 30
  3758.6  829.52  3954.4  822.60  4016.3  821.88  4024.0  820.90  4129.6  817.29
  4312.6  812.77  4335.8  812.54  4346.1  813.54  4387.3  810.89  4428.6  811.18
  4449.2  814.93  4459.5  812.48  4766.1  811.02  4771.3  812.10  4789.3  810.93
  4840.9  811.22  4853.8  810.23  4871.8  811.14  4985.2  807.58  4998.5  806.13
  5004.0  802.28  5005.4  801.78  5014.1  802.28  5018.0  802.92  5024.0  805.50
  5031.6  811.09  5039.1  814.33  5054.1  816.38  5117.2  820.53  5175.8  822.49
#Mann=3,-1,0
  3758.6    0.05       0  5004.0   0.033       0  5014.1    0.05       0
Bank Sta=5004,5014.1
Exp/Cntr=0.3,0.1

Type RM Length L Ch R = 1,38425,504,504,504
BEGIN DESCRIPTION:
Morris Branch 62.0
END DESCRIPTION:
XS GIS Cut Line= 3
      2296228.53      7118126.28      2296155.26      7117031.20
      2295878.99      7116709.99
#Sta/Elev= 30
  3931.0  824.56  4107.7  819.96  4157.8  816.99  4207.9  816.23  4227.9  814.94
  4445.8  810.54  4528.6  811.20  4595.9  809.55  4600.9  810.32  4638.9  809.50
  4678.9  810.09  4729.1  809.01  4759.1  807.01  4859.4  808.39  4929.5  807.37
  4979.6  803.66  4984.6  801.64  4986.0  801.14  4994.7  801.64  4999.7  803.13
  5026.6  807.12  5033.6  806.72  5076.4  810.12  5119.2  809.73  5182.8  812.27
  5254.1  813.61  5310.1  817.98  5402.3  822.04  5424.2  822.19  5452.2  824.41
#Mann=3,-1,0
  3931.0    0.05       0  4984.6   0.033       0  4994.7    0.05       0
Bank Sta=4984.6,4994.7
Exp/Cntr=0.3,0.1

Type RM Length L Ch R = 1,37921,500,500,500
BEGIN DESCRIPTION:
Morris Branch 61.0
END DESCRIPTION:
XS GIS Cut Line= 5
      2297101.30      7117725.15      2296829.00      7117260.00
      2296429.00      7116960.00      2296129.00      7116760.00
      2295832.49      7116562.33
#Sta/Elev= 30
  3960.6  819.82  4067.9  818.50  4255.9  816.64  4267.8  816.27  4382.8  813.50
  4649.6  810.37  4671.5  807.76  4699.6  807.72  4736.0  800.72  4799.6  806.04
  4849.6  805.05  4949.6  806.89  4956.9  802.96  4963.1  806.38  4971.5  799.23
  4977.7  799.87  4991.4  797.66  4992.8  797.16  5001.6  797.66  5007.1  800.51
  5079.2  804.91  5085.2  803.43  5115.3  806.06  5280.5  809.03  5301.6  811.28
  5547.9  819.33  5563.0  818.63  5591.7  821.33  5656.1  826.19  5716.5  828.10
#Mann=8,-1,0
  3960.6    0.05       0  4067.9    0.12       0  4255.9    0.05       0
  4267.8    0.12       0  4382.8    0.05       0  4991.4   0.033       0
  5001.6    0.05       0  5591.7   0.075       0
Bank Sta=4991.4,5001.6
Exp/Cntr=0.3,0.1

Type RM Length L Ch R = 1,37421,409,409,409
BEGIN DESCRIPTION:
Morris Branch 60.0
END DESCRIPTION:
XS GIS Cut Line= 4
      2297166.79      7117785.61      2296829.00      7117110.00
      2296635.82      7116686.65      2296280.70      7115960.98
#Sta/Elev= 30
  3804.9  821.96  4067.9  817.69  4167.3  816.76  4261.2  814.39  4277.9  816.03
  4300.3  814.10  4367.4  812.98  4417.7  813.70  4515.5  811.18  4695.2  810.16
  4735.8  808.23  4758.1  803.97  4769.8  799.95  4792.8  797.97  4838.9  800.84
  4959.6  801.68  4967.0  796.36  4972.0  795.17  4973.4  794.67  4982.3  795.17
  5025.6  799.07  5028.6  801.49  5034.2  802.43  5066.4  801.85  5101.7  804.68
  5349.3  805.25  5522.9  809.91  5551.8  812.99  5596.9  823.84  5833.5  831.88
#Mann=5,-1,0
  3804.9    0.05       0  4067.9    0.12       0  4167.3    0.05       0
  4972.0   0.033       0  4982.3    0.05       0
Bank Sta=4972,4982.3
Exp/Cntr=0.3,0.1

Type RM Length L Ch R = 1,37012,468,468,468
BEGIN DESCRIPTION:
Morris Branch 59.0
END DESCRIPTION:
XS GIS Cut Line= 4
      2297276.51      7117674.98      2296879.00      7116960.00
      2296929.00      7116460.00      2296321.00      7115867.93
#Sta/Elev= 30
  3686.9  821.92  4166.4  814.67  4231.6  812.69  4350.5  811.66  4356.3  812.64
  4372.3  811.31  4431.8  811.71  4453.5  810.29  4475.2  811.26  4535.1  810.41
  4854.2  799.67  4896.9  799.17  4917.0  801.17  4977.3  798.52  4999.4  795.63
  5000.9  795.13  5010.5  795.63  5014.5  795.65  5021.5  799.71  5028.7  799.99
  5035.6  802.84  5198.4  802.54  5410.6  805.89  5516.6  812.93  5580.2  814.95
  5672.2  820.24  5707.5  820.88  5714.6  822.15  5834.8  825.28  5856.1  827.96
#Mann=3,-1,0
  3686.9    0.05       0  4999.4   0.033       0  5010.5    0.05       0
Bank Sta=4999.4,5010.5
Exp/Cntr=0.3,0.1

Type RM Length L Ch R = 1,36544,414,414,414
BEGIN DESCRIPTION:
Morris Branch 58.0
END DESCRIPTION:
XS GIS Cut Line= 3
      2297578.98      7117159.96      2297329.00      7116460.00
      2297179.00      7115660.00
#Sta/Elev= 30
  4247.3  819.04  4293.4  817.07  4349.7  810.45  4491.5  803.52  4616.3  801.66
  4926.8  801.26  4937.5  800.78  4949.7  795.76  5056.2  795.47  5057.7  794.97
  5067.3  795.47  5102.5  800.82  5163.5  800.29  5204.2  795.95  5237.3  796.71
  5284.8  795.59  5295.8  799.05  5306.0  799.40  5336.5  797.45  5347.5  799.34
  5428.1  802.14  5447.6  800.65  5499.3  801.65  5550.1  806.08  5615.4  821.65
  5621.4  824.26  5668.0  832.37  5700.2  836.24  5720.6  839.29  5804.5  846.61
#Mann=4,-1,0
  4247.3    0.05       0  5056.2   0.033       0  5067.3    0.05       0
  5700.2    0.05       0
Bank Sta=5056.2,5067.3
Exp/Cntr=0.3,0.1

Type RM Length L Ch R = 1,36130,431,431,431
BEGIN DESCRIPTION:
Morris Branch 57.0
END DESCRIPTION:
XS GIS Cut Line= 3
      2297629.00      7117110.04      2297629.00      7116210.00
      2297329.02      7115810.03
#Sta/Elev= 30
  4105.0  817.99  4145.0  815.64  4175.0  809.79  4205.0  806.47  4295.0  801.27
  4505.0  799.04  4675.0  799.33  4785.0  797.23  4915.0  799.53  4945.0  798.80
  4969.3  795.84  4970.9  795.34  4980.7  795.84  5026.9  797.67  5047.7  796.41
  5062.3  798.76  5133.2  798.22  5141.5  799.75  5147.7  797.33  5153.7  798.27
  5162.3  800.14  5176.9  798.20  5212.3  798.20  5305.0  800.24  5347.7  804.22
  5376.9  810.08  5383.2  809.43  5405.0  816.40  5424.5  818.33  5505.0  827.87
#Mann=5,-1,0
  4105.0    0.05       0  4969.3   0.033       0  4980.7    0.05       0
  5153.7    0.12       0  5424.5    0.05       0
Bank Sta=4969.3,4980.7
Exp/Cntr=0.3,0.1
