HEC-RAS study Morris Branch.prj: Morris Branch Base Level Engineering

--- Morris Branch.g01 (geometry) --- (continued)

Type RM Length L Ch R = 1,35699,471,471,471
BEGIN DESCRIPTION:
Morris Branch 56.0
END DESCRIPTION:
XS GIS Cut Line= 3
      2297628.99      7117210.03      2298029.00      7116110.00
      2297628.99      7115709.99
#Sta/Elev= 30
  3833.6  820.73  3910.1  819.10  3966.0  817.26  3991.2  814.71  3996.6  815.16
  4021.8  809.03  4027.2  808.80  4052.4  805.09  4077.7  802.96  4108.3  801.21
  4163.5  800.33  4169.5  799.43  4291.8  798.18  4397.6  797.86  4459.4  796.53
  5131.4  796.51  5224.7  795.26  5226.2  794.76  5234.5  794.76  5236.1  795.26
  5258.7  795.27  5272.8  796.18  5315.2  797.00  5329.4  798.15  5385.9  799.97
  5442.5  803.76  5484.9  808.46  5513.2  814.30  5541.5  815.98  5569.8  818.57
#Mann=3,-1,0
  3833.6    0.05       0  5224.7   0.033       0  5236.1    0.05       0
Bank Sta=5224.7,5236.1
Exp/Cntr=0.3,0.1

Type RM Length L Ch R = 1,35228,437,437,437
BEGIN DESCRIPTION:
Morris Branch 55.0
END DESCRIPTION:
XS GIS Cut Line= 3
      2297728.99      7117210.01      2298429.00      7116010.00
      2298479.00      7115210.02
#Sta/Elev= 30
  3617.9  820.22  3749.0  817.42  3770.5  815.61  3786.2  812.51  3807.7  811.01
  3814.7  809.16  3837.9  807.12  3844.9  805.31  3866.4  804.71  3882.1  802.64
  3887.9  803.09  3918.9  800.63  3999.5  798.60  4173.6  796.25  4304.7  795.62
  5322.0  795.00  5323.6  794.50  5333.6  795.00  5357.8  795.55  5367.9  797.19
  5377.9  799.47  5387.9  804.27  5405.4  807.52  5410.4  806.91  5468.1  812.46
  5478.1  815.07  5488.1  816.30  5731.1  837.44  5758.6  841.44  5808.7  845.68
#Mann=3,-1,0
  3617.9    0.05       0  5322.0   0.033       0  5333.6    0.05       0
Bank Sta=5322,5333.6
Exp/Cntr=0.3,0.1

Type RM Length L Ch R = 1,34791,678,678,678
BEGIN DESCRIPTION:
Morris Branch 54.0
END DESCRIPTION:
XS GIS Cut Line= 3
      2299129.00      7117309.99      2298829.00      7116110.00
      2298678.99      7115309.97
#Sta/Elev= 30
  3763.9  818.76  3846.4  818.00  3864.4  816.17  3959.7  814.54  3988.1  813.41
  4153.0  809.63  4359.2  801.54  4488.0  797.24  4516.4  795.81  4518.3  795.01
  4519.9  794.51  4528.3  794.51  4529.9  795.01  5448.5  795.27  5489.2  800.57
  5509.5  802.16  5515.5  803.51  5540.1  804.98  5550.2  807.57  5568.0  809.71
  5601.1  812.51  5641.8  817.96  5713.0  824.79  5730.8  827.58  5735.9  826.78
  5763.9  830.77  5783.4  832.45  5788.5  832.04  5794.4  833.38  5814.8  835.00
#Mann=3,-1,0
  3763.9    0.05       0  4518.3   0.033       0  4529.9    0.05       0
Bank Sta=4518.3,4529.9
Exp/Cntr=0.3,0.1

Type RM Length L Ch R = 1,34113,132,132,132
BEGIN DESCRIPTION:
Mapping XS 6bba3084
END DESCRIPTION:
XS GIS Cut Line= 6
      2299783.25      7117786.22      2299701.61      7116485.34
      2299285.33      7115554.70      2299024.27      7115456.78
      2298782.99      7115558.19      2298680.73      7115236.79
#Sta/Elev= 30
  2901.5  824.12  3669.2  808.29  3705.1  803.73  4060.0  797.65  4070.0  795.08
  4485.8  794.72  4487.4  794.22  4497.4  794.72  5500.5  795.44  5560.7  800.42
  5589.8  799.01  5613.6  802.44  5619.0  800.64  5637.3  803.58  5666.5  802.33
  5737.8  806.83  5743.2  804.84  5766.9  807.93  5776.5  805.90  5804.0  811.46
  5873.7  818.56  5900.7  818.37  5906.0  820.79  5938.2  819.27  5943.4  823.25
  6002.6  824.50  6007.9  827.72  6034.9  827.81  6040.1  831.89  6114.3  839.60
#Mann=3,-1,0
  2901.5    0.05       0  4485.8   0.033       0  4497.4    0.05       0
Bank Sta=4485.8,4497.4
Exp/Cntr=0.3,0.1

Type RM Length L Ch R = 1,33981,100,100,100
BEGIN DESCRIPTION:
Mapping XS 1035d466
END DESCRIPTION:
XS GIS Cut Line= 6
      2299835.54      7117775.21      2299795.80      7116430.87
      2299323.42      7115390.60      2299240.56      7115307.50
      2299087.92      7115284.28      2298970.95      7114980.11
#Sta/Elev= 30
  2923.4  826.22  3598.7  811.22  3878.7  815.62  3884.1  815.57  3889.1  812.44
  4174.6  816.47  4179.7  813.94  4226.3  816.45  4231.4  814.76  4597.5  817.23
  4908.9  815.69  4937.9  817.37  4985.0  815.56  5037.7  817.19  5061.2  815.14
  5066.7  817.22  5107.4  815.74  5388.3  816.78  5438.2  816.21  5445.3  814.31
  5494.8  816.31  5679.8  815.90  5695.6  812.59  5720.3  811.38  5889.1  811.03
  5890.7  810.53  5900.7  811.03  5925.5  811.82  5968.4  821.08  6011.1  819.43
#Mann=3,-1,0
  2923.4    0.05       0  5889.1   0.033       0  5900.7    0.05       0
Bank Sta=5889.1,5900.7
Exp/Cntr=0.3,0.1

Type RM Length L Ch R = 1,33881,790,790,790
BEGIN DESCRIPTION:
Mapping XS f28ee07c
END DESCRIPTION:
XS GIS Cut Line= 4
      2300161.17      7116938.25      2299984.72      7116561.85
      2299464.74      7115452.65      2299797.85      7114915.02
#Sta/Elev= 30
  3698.7  807.33  3720.0  805.23  3760.1  803.58  3917.6  799.20  3971.0  796.23
  4016.7  796.73  4022.2  797.78  4096.2  797.26  4182.0  795.31  4210.3  793.45
  4337.3  790.99  4414.6  787.50  4609.4  785.26  4768.9  784.89  4770.5  784.39
  4780.5  784.89  5143.6  785.73  5219.4  786.86  5395.2  792.44  5410.6  791.36
  5416.5  789.64  5437.8  789.54  5657.5  793.44  5678.8  792.39  5715.4  797.02
  5742.6  802.19  5801.3  805.71  5889.1  814.33  5941.1  817.95  5971.9  821.66
#Mann=3,-1,0
  3698.7    0.05       0  4768.9   0.033       0  4780.5    0.05       0
Bank Sta=4768.9,4780.5
Exp/Cntr=0.3,0.1

Type RM Length L Ch R = 1,33091,307,307,307
BEGIN DESCRIPTION:
Mapping XS abfa5532
END DESCRIPTION:
XS GIS Cut Line= 2
      2300160.29      7116126.44      2300200.03      7115096.61
#Sta/Elev= 30
  4440.9  786.82  4567.4  784.90  4577.4  785.31  4597.5  783.68  4617.5  783.23
  4707.5  782.82  4727.6  783.53  4767.6  783.41  4827.6  781.81  4927.7  781.76
  4957.7  779.41  4987.8  780.40  5017.8  773.89  5041.8  771.97  5043.5  771.47
  5053.7  771.97  5054.3  778.44  5067.8  782.48  5107.8  781.64  5137.9  782.41
  5197.9  782.13  5227.9  782.96  5247.9  782.37  5348.0  784.11  5358.0  786.03
  5378.0  791.57  5418.1  804.50  5428.1  805.17  5438.1  807.87  5471.5  811.58
#Mann=3,-1,0
  4440.9    0.05       0  5041.8   0.033       0  5053.7    0.05       0
Bank Sta=5041.8,5053.7
Exp/Cntr=0.3,0.1

Type RM Length L Ch R = 1,32784,534,534,534
BEGIN DESCRIPTION:
Mapping XS 1bf8d6a4
END DESCRIPTION:
XS GIS Cut Line= 3
      2300492.41      7116039.00      2300457.19      7115220.48
      2300442.29      7114874.27
#Sta/Elev= 30
  4568.1  784.47  4707.2  781.27  4967.5  780.49  4977.5  779.83  4994.4  774.09
  4999.4  774.63  5001.5  770.97  5003.2  770.47  5013.5  770.97  5017.5  771.17
  5027.5  774.37  5087.6  777.14  5117.6  780.30  5167.6  781.32  5257.7  779.80
  5267.7  780.74  5287.8  779.88  5307.8  780.64  5327.8  779.51  5347.8  780.71
  5357.8  779.80  5427.9  781.09  5487.9  783.12  5531.5  789.35  5568.0  795.61
  5588.0  801.63  5598.0  806.13  5658.1  814.96  5678.1  816.02  5733.9  824.65
#Mann=4,-1,0
  4568.1    0.05       0  5001.5   0.035       0  5013.5    0.05       0
  5531.5    0.12       0
Bank Sta=5001.5,5013.5
Exp/Cntr=0.3,0.1

Type RM Length L Ch R = 1,32250,713,713,713
BEGIN DESCRIPTION:
Mapping XS ac4c092d
END DESCRIPTION:
XS GIS Cut Line= 3
      2301123.92      7115863.71      2300614.67      7115126.87
      2300440.34      7114874.64
#Sta/Elev= 30
  4658.1  784.33  4808.5  783.41  4881.0  778.24  4973.8  777.89  4988.4  778.34
  4994.5  771.77  5003.0  771.08  5009.4  768.45  5009.5  766.72  5011.1  766.22
  5021.5  766.72  5039.1  768.61  5045.2  771.01  5060.1  771.09  5066.2  773.19
  5075.0  773.74  5095.9  777.82  5215.7  778.64  5233.1  779.25  5340.6  777.26
  5382.5  778.67  5534.6  779.53  5636.4  781.43  5683.9  787.99  5692.7  790.86
  5698.8  795.67  5713.7  801.07  5756.6  809.96  5815.1  817.27  5860.4  824.65
#Mann=6,-1,0
  4658.1    0.05       0  4973.8    0.12       0  5009.5    0.07       0
  5021.5    0.12       0  5215.7    0.05       0  5636.4    0.12       0
Bank Sta=5009.5,5021.5
Exp/Cntr=0.3,0.1

Type RM Length L Ch R = 1,31537,698,698,698
BEGIN DESCRIPTION:
Mapping XS 3cb856cd
END DESCRIPTION:
XS GIS Cut Line= 2
      2301410.71      7115585.30      2301114.33      7114704.21
#Sta/Elev= 30
  4442.3  778.31  4621.1  775.40  4954.3  775.61  4962.4  774.96  4973.8  769.14
  4979.9  764.73  4981.6  764.23  4992.0  764.73  4999.2  766.93  5017.6  767.60
  5030.7  770.09  5056.9  771.42  5062.2  772.50  5070.4  769.88  5080.9  773.05
  5088.4  774.05  5119.9  775.29  5125.2  776.24  5144.2  775.75  5165.3  776.78
  5207.5  776.65  5214.5  777.76  5270.8  778.18  5277.5  780.57  5282.8  779.51
  5302.5  783.71  5314.3  784.94  5330.4  789.58  5340.5  792.49  5371.9  793.78
#Mann=5,-1,0
  4442.3    0.05       0  4973.8    0.12       0  4979.9    0.07       0
  4992.0    0.12       0  5330.4    0.05       0
Bank Sta=4979.9,4992
Exp/Cntr=0.3,0.1

Type RM Length L Ch R = 1,30839,1310,1310,1310
BEGIN DESCRIPTION:
Mapping XS 5e4065bc
END DESCRIPTION:
XS GIS Cut Line= 2
      2301937.14      7115365.66      2301478.85      7114278.72
#Sta/Elev= 30
  4417.0  776.31  4466.5  776.45  4479.7  778.96  4503.4  771.86  4527.1  771.04
  4632.9  771.77  4780.6  770.13  4957.4  771.50  4986.7  767.07  4992.1  764.56
  5015.8  764.48  5024.8  763.10  5026.5  762.60  5036.9  763.10  5045.0  765.37
  5063.3  764.98  5068.7  767.07  5074.3  764.27  5085.1  772.59  5092.4  774.56
  5116.2  774.72  5121.6  772.66  5192.7  777.80  5322.2  781.75  5345.6  781.31
  5456.4  789.48  5486.7  794.08  5557.4  796.95  5562.8  798.44  5596.6  800.64
#Mann=5,-1,0
  4417.0    0.05       0  4957.4    0.12       0  5024.8    0.07       0
  5036.9    0.12       0  5456.4    0.05       0
Bank Sta=5024.8,5036.9
Exp/Cntr=0.3,0.1

Type RM Length L Ch R = 1,29529,730,730,730
BEGIN DESCRIPTION:
Mapping XS b86a04c7
END DESCRIPTION:
XS GIS Cut Line= 2
      2302319.74      7115326.31      2302288.83      7114447.26
#Sta/Elev= 30
  4655.0  773.98  4671.3  775.13  4681.3  772.93  4751.4  770.10  4831.4  770.59
  4951.5  768.19  4971.5  765.89  4991.5  760.56  4995.4  757.70  4997.1  757.20
  5007.6  757.70  5021.5  758.59  5028.1  759.92  5051.6  763.88  5061.6  767.72
  5071.6  768.29  5141.6  767.43  5151.6  768.00  5231.7  767.81  5251.7  769.31
  5321.7  771.31  5341.7  773.23  5361.7  774.09  5381.8  776.57  5387.1  779.22
  5392.1  778.90  5401.8  780.89  5461.8  796.72  5501.8  802.93  5534.6  806.70
#Mann=4,-1,0
  4655.0    0.05       0  4995.4   0.035       0  5007.6    0.05       0
  5028.1    0.12       0
Bank Sta=4995.4,5007.6
Exp/Cntr=0.3,0.1

Type RM Length L Ch R = 1,28799,384,384,384
BEGIN DESCRIPTION:
Mapping XS cc78b42d
END DESCRIPTION:
XS GIS Cut Line= 3
      2302695.33      7115260.96      2302697.59      7114693.95
      2302639.22      7114355.67
#Sta/Elev= 30
  4296.9  772.48  4467.9  766.14  4537.9  765.57  4587.9  766.59  4657.9  765.31
  4677.9  766.43  4737.9  765.76  4765.7  766.70  4797.9  766.38  4807.9  767.61
  4837.9  765.56  4868.5  765.83  4898.4  761.97  4943.9  760.94  4949.1  759.90
  4959.3  760.08  4969.4  758.20  4989.7  758.74  5010.0  757.12  5014.0  755.21
  5015.7  754.71  5026.3  755.21  5030.3  759.07  5050.6  769.13  5063.6  773.47
  5123.5  777.11  5163.0  780.85  5172.4  781.96  5192.7  787.13  5207.2  788.12
#Mann=5,-1,0
  4296.9    0.05       0  4765.7    0.12       0  5014.0    0.07       0
  5026.3    0.12       0  5163.0    0.05       0
Bank Sta=5014,5026.3
Exp/Cntr=0.3,0.1

Type RM Length L Ch R = 1,28415,646,646,646
BEGIN DESCRIPTION:
Mapping XS faf1ad4d
END DESCRIPTION:
XS GIS Cut Line= 2
      2303011.70      7115290.24      2303061.67      7114334.54
#Sta/Elev= 30
  4246.5  769.49  4467.0  764.64  4597.2  763.75  4647.3  764.95  4663.4  764.35
  4697.4  763.95  4707.4  762.75  4727.4  764.44  4737.4  759.31  4747.4  756.62
  4757.4  762.10  4777.5  765.37  4797.5  763.52  4847.6  762.30  4897.6  764.93
  4937.7  762.84  4947.7  763.12  4977.7  759.96  4997.8  755.13  5011.6  753.06
  5013.3  752.56  5023.9  753.06  5027.8  755.21  5037.8  757.85  5054.7  767.16
  5067.9  772.68  5097.9  779.52  5144.5  787.28  5158.0  788.81  5203.5  796.94
#Mann=5,-1,0
  4246.5    0.05       0  4663.4    0.12       0  5011.6    0.07       0
  5023.9    0.12       0  5144.5    0.05       0
Bank Sta=5011.6,5023.9
Exp/Cntr=0.3,0.1

Type RM Length L Ch R = 1,27769,337,337,337
BEGIN DESCRIPTION:
Mapping XS 253fc59c
END DESCRIPTION:
XS GIS Cut Line= 2
      2303306.19      7115323.62      2303366.66      7114403.60
#Sta/Elev= 30
  4535.5  764.36  4639.3  763.27  4899.9  762.99  4945.2  763.87  4957.3  762.78
  4962.3  763.52  4970.1  756.06  4973.9  750.30  4975.6  749.80  4986.2  750.30
  5010.1  753.49  5020.2  752.78  5050.2  756.60  5070.3  757.85  5091.3  761.56
  5140.4  764.21  5210.6  766.17  5230.6  765.82  5240.6  766.77  5280.7  766.75
  5320.8  767.81  5340.8  769.98  5350.9  772.24  5360.9  775.80  5370.9  777.34
  5391.0  783.63  5401.0  784.54  5416.5  788.73  5421.5  788.59  5457.5  794.62
#Mann=5,-1,0
  4535.5    0.05       0  4945.2    0.12       0  4973.9    0.07       0
  4986.2    0.12       0  5091.3    0.05       0
Bank Sta=4973.9,4986.2
Exp/Cntr=0.3,0.1

Type RM Length L Ch R = 1,27432,502,502,502
BEGIN DESCRIPTION:
Mapping XS cb957590
END DESCRIPTION:
XS GIS Cut Line= 4
      2303565.70      7115815.47      2303592.45      7115447.81
      2303651.93      7114630.30      2303613.88      7114475.51
#Sta/Elev= 30
  3941.3  768.66  4097.2  763.60  4247.6  760.78  4267.6  761.85  4478.2  759.80
  4588.5  760.18  4728.7  759.25  4744.3  759.63  4779.0  758.22  4878.4  759.45
  4909.3  754.58  4919.4  754.37  4939.4  751.99  4996.4  750.60  5003.4  749.37
  5005.1  748.87  5015.7  749.37  5017.4  754.12  5022.5  751.46  5029.6  758.99
  5039.7  760.95  5079.8  762.55  5099.8  764.31  5109.9  766.53  5164.4  768.85
  5205.9  771.47  5222.6  774.25  5242.3  775.46  5263.8  777.92  5289.0  781.78
#Mann=5,-1,0
  3941.3    0.05       0  4728.7    0.12       0  4996.4    0.05       0
  5003.4   0.033       0  5015.7    0.05       0
Bank Sta=5003.4,5015.7
Exp/Cntr=0.3,0.1

Type RM Length L Ch R = 1,26930,539,539,539
BEGIN DESCRIPTION:
Mapping XS 2a7f42ed
END DESCRIPTION:
XS GIS Cut Line= 3
      2303774.54      7115862.12      2303871.65      7115550.29
      2304157.29      7114633.15
#Sta/Elev= 30
  4055.4  763.65  4388.7  758.41  4453.8  759.23  4659.4  757.50  4707.8  758.79
  4724.5  757.99  4729.7  754.77  4738.4  753.49  4762.2  752.14  4811.7  753.61
  4832.7  757.94  4924.8  758.92  4947.9  752.64  4961.6  751.56  4984.4  749.73
  5000.4  748.36  5004.5  746.07  5006.3  745.57  5016.9  746.07  5032.9  749.22
  5052.6  756.74  5065.4  758.78  5178.3  761.34  5220.2  764.25  5232.0  766.39
  5251.6  769.23  5265.8  773.89  5283.1  776.07  5304.0  782.76  5342.6  784.86
#Mann=7,-1,0
  4055.4    0.05       0  4707.8    0.12       0  4961.6    0.05       0
  4984.4    0.12       0  5004.5    0.07       0  5016.9    0.12       0
  5232.0    0.05       0
Bank Sta=5004.5,5016.9
Exp/Cntr=0.3,0.1

Type RM Length L Ch R = 1,26391,1041,1041,1041
BEGIN DESCRIPTION:
Mapping XS d54dee83
END DESCRIPTION:
XS GIS Cut Line= 3
      2303980.37      7115665.70      2304455.30      7115151.21
      2304642.02      7114628.55
#Sta/Elev= 30
  4042.8  757.84  4243.9  757.16  4273.2  758.15  4336.3  757.74  4418.8  755.04
  4442.3  752.17  4505.8  751.39  4555.2  753.24  4576.7  755.61  4635.0  754.80
  4795.3  755.50  4818.6  753.76  4839.8  749.89  4850.5  750.01  4856.9  751.78
  4903.6  750.43  4944.0  745.18  4974.7  745.89  4992.9  743.02  4994.7  742.52
  5005.3  743.02  5005.5  751.74  5010.8  751.31  5020.4  756.67  5105.6  757.49
  5203.3  760.66  5254.0  762.17  5272.0  764.72  5277.3  763.20  5298.0  765.86
#Mann=8,-1,0
  4042.8    0.05       0  4273.2    0.12       0  4418.8    0.05       0
  4635.0    0.12       0  4992.9    0.07       0  5005.3    0.12       0
  5105.6    0.05       0  5203.3    0.12       0
Bank Sta=4992.9,5005.3
Exp/Cntr=0.3,0.1

Type RM Length L Ch R = 1,25350,824,824,824
BEGIN DESCRIPTION:
Mapping XS e24f6305
END DESCRIPTION:
XS GIS Cut Line= 3
      2305092.44      7115947.57      2305057.82      7115455.17
      2304985.54      7114569.73
#Sta/Elev= 30
  4460.9  763.34  4618.9  762.09  4648.9  763.88  4659.0  763.21  4669.0  760.10
  4729.1  759.92  4749.2  757.04  4759.2  752.96  4769.2  750.89  4779.3  745.81
  4789.3  742.32  4799.3  741.01  4809.3  747.31  4819.4  750.38  4829.4  749.99
  4865.4  752.36  4959.7  751.76  4969.7  751.23  4989.8  739.44  5009.9  739.43
  5013.7  737.55  5015.5  737.05  5026.1  737.55  5050.0  749.66  5060.0  752.00
  5137.8  750.98  5361.0  750.23  5712.2  753.83  5743.1  756.64  5842.9  761.15
#Mann=4,-1,0
  4460.9    0.05       0  5013.7   0.033       0  5026.1    0.05       0
  5137.8    0.05       0
Bank Sta=5013.7,5026.1
Exp/Cntr=0.3,0.1

Type RM Length L Ch R = 1,24526,461,461,461
BEGIN DESCRIPTION:
Morris Branch 38.0
END DESCRIPTION:
XS GIS Cut Line= 3
      2305828.99      7115759.98      2305529.00      7114860.00
      2305378.98      7114509.96
#Sta/Elev= 30
  4055.7  758.93  4256.0  754.04  4277.0  755.30  4298.1  753.68  4340.3  753.93
  4393.0  750.34  4498.4  749.91  4572.2  747.49  4688.1  746.73  4730.3  749.56
  4920.0  746.94  4930.6  746.13  4941.1  741.44  4962.2  735.78  4976.2  734.98
  4978.2  734.48  4990.4  734.98  5001.7  738.50  5013.4  739.17  5028.0  744.12
  5047.9  747.78  5066.0  748.61  5135.6  748.32  5215.4  749.00  5243.1  749.24
  5287.2  750.70  5299.9  753.63  5323.5  754.67  5363.4  772.20  5385.2  775.12
#Mann=7,-1,0
  4055.7    0.05       0  4976.2   0.033       0  4990.4    0.05       0
  5028.0    0.12       0  5135.6    0.05       0  5215.4    0.12       0
  5243.1    0.05       0
Bank Sta=4976.2,4990.4
Exp/Cntr=0.3,0.1

Type RM Length L Ch R = 1,24065,400,400,400
BEGIN DESCRIPTION:
Morris Branch 37.0
END DESCRIPTION:
XS GIS Cut Line= 3
      2306379.02      7115410.04      2305879.00      7114610.00
      2305428.99      7114460.00
#Sta/Elev= 30
  4048.9  756.66  4172.2  755.64  4245.3  750.75  4296.6  749.83  4318.4  744.50
  4337.8  743.96  4362.7  742.99  4382.1  742.72  4403.3  745.84  4449.3  744.33
  4543.6  745.80  4790.1  744.21  4911.6  745.25  4926.9  744.86  4942.2  739.92
  4956.7  737.80  4978.8  735.13  5002.9  735.97  5016.9  733.11  5018.9  732.61
  5031.1  733.11  5045.0  739.44  5055.6  741.91  5087.2  745.11  5217.1  748.01
  5350.7  752.08  5414.0  758.54  5445.6  766.42  5456.1  772.24  5466.7  774.27
#Mann=7,-1,0
  4048.9    0.05       0  4337.8    0.12       0  4362.7    0.05       0
  4956.7    0.12       0  5016.9    0.07       0  5031.1    0.12       0
  5217.1    0.05       0
#XS Ineff=2,0
    0.00 4750.00  760.45               0
Permanent Ineff=
       F       F
Bank Sta=5016.9,5031.1
Exp/Cntr=0.3,0.1

Type RM Length L Ch R = 1,23665,386,386,386
BEGIN DESCRIPTION:
Mapping XS b9833af2
END DESCRIPTION:
XS GIS Cut Line= 2
      2306397.62      7114829.69      2306059.40      7114107.57
#Sta/Elev= 30
  4557.8  749.96  4661.5  748.52  4678.8  747.01  4684.3  748.04  4690.0  745.33
  4699.6  743.31  4730.0  742.76  4745.2  740.01  4775.7  738.23  4826.8  743.18
  4859.2  742.56  4902.1  741.59  4986.7  741.65  4992.2  740.81  4999.2  738.02
  5009.5  736.40  5014.1  731.37  5016.1  730.87  5028.3  731.37  5054.4  735.28
  5076.5  736.25  5089.0  740.77  5120.6  744.12  5209.0  745.62  5220.0  746.16
  5226.0  747.47  5231.5  746.63  5242.1  746.77  5280.1  748.72  5355.2  752.31
#Mann=7,-1,0
  4557.8    0.05       0  4699.6    0.12       0  4859.2    0.05       0
  4902.1    0.12       0  5014.1    0.07       0  5028.3    0.12       0
  5280.1    0.05       0
Bank Sta=5014.1,5028.3
Exp/Cntr=0.3,0.1

Type RM Length L Ch R = 1,23279,204,204,204
BEGIN DESCRIPTION:
Mapping XS 000cd0bb
END DESCRIPTION:
XS GIS Cut Line= 2
      2306649.87      7114724.09      2306370.17      7113976.61
#Sta/Elev= 30
  4451.2  744.20  4519.6  742.97  4525.0  745.50  4549.9  745.73  4604.5  741.87
  4687.2  737.20  4696.0  734.13  4711.8  735.99  4721.0  740.96  4733.2  741.56
  4850.6  739.69  4946.7  741.12  4968.1  736.20  5012.4  731.67  5014.3  730.37
  5016.3  729.87  5028.6  730.37  5053.5  731.75  5063.0  735.64  5068.3  740.79
  5074.8  742.44  5093.3  740.01  5098.6  743.20  5106.9  741.34  5123.6  748.44
  5128.9  748.32  5153.8  754.79  5187.5  757.89  5209.1  768.43  5249.3  768.41
#Mann=7,-1,0
  4451.2    0.05       0  4604.5    0.12       0  4687.2    0.05       0
  5012.4    0.12       0  5014.3   0.033       0  5028.6    0.12       0
  5187.5    0.05       0
Bank Sta=5014.3,5028.6
Exp/Cntr=0.3,0.1

Type RM Length L Ch R = 1,23075,192,192,192
BEGIN DESCRIPTION:
Mapping XS 98db263d
END DESCRIPTION:
XS GIS Cut Line= 3
      2306938.55      7114868.29      2306864.98      7114691.74
      2306513.74      7113848.86
#Sta/Elev= 30
  4145.2  745.80  4259.1  743.89  4424.8  745.22  4497.3  742.47  4511.7  741.21
  4524.5  736.63  4548.3  732.27  4565.9  736.65  4596.0  737.09  4619.8  741.07
  4702.1  741.38  4707.5  739.51  4938.3  739.90  4955.9  737.21  4967.5  732.74
  4991.8  730.66  4992.0  730.57  4994.0  730.07  5006.3  730.57  5020.9  734.74
  5075.0  734.64  5085.9  736.38  5092.1  740.37  5115.9  745.24  5129.2  751.40
  5139.8  753.57  5150.9  759.83  5166.8  762.78  5192.9  769.36  5249.6  771.27
#Mann=7,-1,0
  4145.2    0.05       0  4424.8    0.12       0  4497.3    0.05       0
  4991.8    0.12       0  4992.0    0.07       0  5006.3    0.12       0
  5166.8    0.05       0
Bank Sta=4992,5006.3
Exp/Cntr=0.3,0.1

Type RM Length L Ch R = 1,22883,463,463,463
BEGIN DESCRIPTION:
Mapping XS 61771269
END DESCRIPTION:
XS GIS Cut Line= 3
      2307181.10      7114694.13      2307052.83      7114481.61
      2306616.36      7113758.45
#Sta/Elev= 30
  4135.8  745.70  4359.6  741.95  4409.4  742.88  4476.0  740.55  4491.0  736.85
  4497.4  732.30  4526.1  736.13  4549.4  736.27  4598.3  740.38  4701.3  738.45
  4730.3  735.83  4751.7  738.29  4788.5  737.06  4920.5  739.62  4957.4  735.83
  4971.6  728.46  4973.6  727.96  4985.9  728.46  5015.6  732.95  5051.7  733.66
  5079.7  737.20  5110.1  742.30  5124.9  746.90  5159.3  754.36  5174.8  754.17
  5180.6  757.08  5190.3  758.30  5203.5  765.00  5217.5  768.73  5228.7  768.94
#Mann=5,-1,0
  4135.8    0.05       0  4409.4    0.12       0  4971.6    0.07       0
  4985.9    0.12       0  5124.9    0.05       0
Bank Sta=4971.6,4985.9
Exp/Cntr=0.3,0.1

Type RM Length L Ch R = 1,22420,590,590,590
BEGIN DESCRIPTION:
Mapping XS 5fb468cd
END DESCRIPTION:
XS GIS Cut Line= 2
      2307428.24      7114437.99      2306954.08      7113489.28
#Sta/Elev= 30
  4084.9  742.12  4180.8  741.44  4359.7  737.82  4404.4  738.63  4426.8  737.79
  4507.5  738.19  4717.5  736.88  4762.2  738.24  4775.8  734.59  4777.3  733.60
  4784.6  728.78  4806.9  732.12  4829.3  732.83  4834.9  735.84  4887.6  736.49
  4946.7  734.73  4963.5  737.54  4977.0  734.75  4991.4  729.31  5023.2  728.29
  5025.2  727.79  5037.9  728.29  5058.5  735.64  5066.4  736.19  5075.3  738.89
  5088.8  747.56  5097.7  751.42  5111.2  754.41  5128.0  754.54  5145.5  753.90
#Mann=5,-1,0
  4084.9    0.05       0  4777.3    0.12       0  5023.2    0.07       0
  5037.9    0.12       0  5128.0    0.05       0
Bank Sta=5023.2,5037.9
Exp/Cntr=0.3,0.1

Type RM Length L Ch R = 1,21830,510,510,510
BEGIN DESCRIPTION:
Mapping XS 2b013c8b
END DESCRIPTION:
XS GIS Cut Line= 3
      2308034.26      7114266.84      2307469.75      7113260.96
      2307141.61      7112963.13
#Sta/Elev= 30
  3844.4  741.59  3986.0  737.66  4191.4  734.20  4528.8  733.81  4661.5  731.71
  4720.8  732.50  4769.9  735.51  4785.8  734.03  4791.4  730.80  4807.5  725.20
  4815.5  727.84  4838.4  730.15  4866.8  735.03  4872.8  734.54  4888.5  729.61
  4926.1  728.41  4931.9  729.29  4969.5  729.54  4985.5  726.55  5001.7  725.79
  5005.5  724.10  5007.5  723.60  5020.3  724.10  5034.6  727.51  5041.3  732.14
  5055.5  734.95  5062.9  735.71  5081.5  734.63  5352.8  738.77  5441.0  741.87
#Mann=5,-1,0
  3844.4    0.05       0  4791.4    0.12       0  5005.5    0.07       0
  5020.3    0.12       0  5081.5    0.05       0
Bank Sta=5005.5,5020.3
Exp/Cntr=0.3,0.1

Type RM Length L Ch R = 1,21320,1027,1027,1027
BEGIN DESCRIPTION:
Mapping XS 53707c23
END DESCRIPTION:
XS GIS Cut Line= 2
      2308384.04      7113893.99      2307446.80      7112330.02
#Sta/Elev= 30
  3951.1  738.08  3993.3  735.33  4177.3  730.85  4491.0  730.34  4512.4  726.20
  4533.8  724.35  4549.4  724.81  4570.8  728.44  4634.9  730.97  4730.2  730.49
  4905.2  732.79  4947.9  726.69  4970.0  727.49  5014.4  722.10  5016.4  721.60
  5029.3  722.10  5043.2  727.94  5058.8  729.35  5144.9  728.04  5196.8  730.70
  5256.9  730.65  5333.2  729.31  5350.4  727.39  5371.8  730.78  5482.6  732.70
  5576.2  738.06  5663.4  746.65  5692.8  758.16  5721.7  759.49  5774.4  765.29
#Mann=5,-1,0
  3951.1    0.05       0  5014.4   0.033       0  5029.3    0.05       0
  5256.9    0.12       0  5333.2    0.05       0
Bank Sta=5014.4,5029.3
Exp/Cntr=0.3,0.1

Type RM Length L Ch R = 1,20293,671,671,671
BEGIN DESCRIPTION:
Mapping XS 51259c8d
END DESCRIPTION:
XS GIS Cut Line= 2
      2308470.57      7113626.46      2308145.37      7112193.50
#Sta/Elev= 30
  3698.1  736.47  3899.6  728.14  3949.7  727.34  4084.1  729.44  4089.3  729.24
  4094.4  726.99  4104.6  725.30  4114.9  724.64  4125.2  726.22  4350.7  728.68
  4371.3  727.66  4576.3  728.59  4730.2  727.46  4884.0  724.37  4906.1  725.96
  4949.2  725.80  4966.0  727.62  4992.3  724.40  4997.2  724.98  5017.3  717.03
  5027.5  717.96  5033.1  716.86  5035.1  716.36  5048.0  716.86  5068.5  732.44
  5078.5  744.01  5083.6  745.48  5089.1  749.91  5156.8  750.69  5167.5  751.04
#Mann=5,-1,0
  3698.1    0.05       0  4997.2    0.12       0  5033.1    0.07       0
  5048.0    0.12       0  5156.8    0.05       0
Bank Sta=5033.1,5048
Exp/Cntr=0.3,0.1

Type RM Length L Ch R = 1,19622,611,611,611
BEGIN DESCRIPTION:
Mapping XS 4f5512ef
END DESCRIPTION:
XS GIS Cut Line= 2
      2309084.18      7113001.79      2308594.40      7112049.34
#Sta/Elev= 30
  4296.7  732.18  4361.6  728.58  4523.6  724.34  4726.0  724.57  4783.0  722.94
  4866.1  724.29  4927.0  722.66  4954.8  724.94  4971.4  724.45  4984.6  717.25
  4986.1  712.44  4988.1  711.94  5001.1  712.44  5015.7  713.22  5021.4  717.05
  5038.1  717.17  5043.5  719.86  5060.1  720.49  5065.7  722.28  5164.6  720.23
  5193.2  720.87  5198.8  722.03  5231.9  721.78  5237.5  722.37  5243.3  725.72
  5254.1  728.12  5259.7  731.23  5288.2  741.35  5322.3  742.06  5367.7  742.27
#Mann=5,-1,0
  4296.7    0.05       0  4986.1   0.033       0  5001.1    0.05       0
  5038.1    0.12       0  5322.3    0.05       0
Bank Sta=4986.1,5001.1
Exp/Cntr=0.3,0.1

Type RM Length L Ch R = 1,19011,372,372,372
BEGIN DESCRIPTION:
Mapping XS 16bad518
END DESCRIPTION:
XS GIS Cut Line= 2
      2309402.02      7112774.51      2308917.73      7111756.43
#Sta/Elev= 30
  4264.7  730.96  4302.0  731.05  4375.7  726.36  4534.7  721.76  4750.2  721.54
  4795.6  719.66  4812.3  717.82  4841.0  720.96  4863.7  721.92  4878.7  722.29
  4900.2  720.79  4923.0  722.44  4945.2  721.78  4954.6  716.00  4967.3  715.76
  4977.3  713.86  4982.9  715.50  4992.5  711.20  4994.5  710.70  5007.5  711.20
  5051.0  716.95  5056.5  715.71  5067.0  718.03  5073.7  721.23  5079.2  720.17
  5111.3  721.41  5119.1  720.93  5124.7  718.48  5199.9  724.87  5392.1  731.26
#Mann=4,-1,0
  4264.7    0.05       0  4900.2    0.12       0  4992.5   0.033       0
  5007.5    0.05       0
Bank Sta=4992.5,5007.5
Exp/Cntr=0.3,0.1

Type RM Length L Ch R = 1,18639,735,735,735
BEGIN DESCRIPTION:
Mapping XS 073ddbb1
END DESCRIPTION:
XS GIS Cut Line= 3
      2309731.51      7112600.55      2309145.84      7111529.43
      2308945.50      7111544.62
#Sta/Elev= 30
  4264.8  734.64  4311.0  734.21  4422.8  727.54  4459.2  727.11  4482.0  723.97
  4591.7  719.48  4657.1  718.44  4771.6  721.00  4826.0  721.38  4842.1  722.73
  4892.3  720.45  4929.4  721.65  4973.0  716.99  5005.3  711.38  5010.1  709.45
  5012.1  708.95  5025.1  709.45  5027.1  712.65  5032.8  714.28  5040.4  718.44
  5048.9  718.80  5063.2  717.86  5086.0  719.89  5255.7  721.11  5326.9  725.16
  5371.0  722.84  5485.6  723.91  5563.5  725.79  5616.6  728.86  5686.5  731.82
#Mann=5,-1,0
  4264.8    0.05       0  4771.6    0.12       0  5010.1    0.07       0
  5025.1    0.12       0  5616.6    0.05       0
Bank Sta=5010.1,5025.1
Exp/Cntr=0.3,0.1

Type RM Length L Ch R = 1,17904,330,330,330
BEGIN DESCRIPTION:
Mapping XS 5c86fe61
END DESCRIPTION:
XS GIS Cut Line= 2
      2310142.62      7112280.26      2309548.80      7110949.32
#Sta/Elev= 30
  4101.8  736.08  4211.6  731.02  4299.7  724.46  4386.8  721.66  4462.3  717.51
  4485.3  717.75  4507.2  716.08  4542.9  717.03  4572.9  716.31  4589.3  717.43
  4635.8  716.71  4791.9  717.88  4868.6  716.06  4884.4  717.81  4907.6  714.85
  4922.0  714.62  4967.2  716.11  5000.0  713.23  5043.8  707.24  5049.4  705.49
  5051.4  704.99  5066.5  705.49  5075.6  720.46  5133.0  719.80  5150.8  718.22
  5268.5  720.26  5394.0  721.39  5445.9  723.55  5474.6  726.00  5559.2  728.20
#Mann=5,-1,0
  4101.8    0.05       0  4922.0    0.12       0  5049.4    0.07       0
  5066.5    0.12       0  5268.5    0.05       0
Bank Sta=5049.4,5066.5
Exp/Cntr=0.3,0.1

Type RM Length L Ch R = 1,17574,326,326,326
BEGIN DESCRIPTION:
Mapping XS 8c971f08
END DESCRIPTION:
XS GIS Cut Line= 2
      2310235.59      7112095.12      2309843.60      7110309.24
#Sta/Elev= 30
  4254.0  728.41  4306.7  724.68  4566.4  716.52  4627.8  716.73  4658.5  714.13
  4682.7  716.22  4726.5  715.13  4791.6  715.47  4819.2  713.83  4868.1  715.39
  4934.8  713.85  4955.4  717.11  4960.8  714.33  4975.9  710.25  4977.6  705.10
  4979.6  704.60  4994.7  705.10  5009.7  706.16  5016.9  711.72  5037.3  713.92
  5053.5  713.10  5078.3  717.53  5109.0  718.15  5139.7  717.05  5609.8  715.78
  5835.9  716.83  5958.8  720.59  6010.0  721.17  6040.7  724.50  6082.4  724.85
#Mann=5,-1,0
  4254.0    0.05       0  4934.8    0.12       0  4977.6    0.07       0
  4994.7    0.12       0  5139.7    0.05       0
Bank Sta=4977.6,4994.7
Exp/Cntr=0.3,0.1

Type RM Length L Ch R = 1,17248,494,494,494
BEGIN DESCRIPTION:
Mapping XS 248e2188
END DESCRIPTION:
XS GIS Cut Line= 3
      2310420.16      7111854.68      2310323.20      7110702.15
      2310054.73      7110125.15
#Sta/Elev= 30
  4412.9  721.87  4638.4  716.70  4718.7  713.79  4729.3  715.03  4758.8  715.82
  4768.8  714.86  4809.0  715.27  4849.2  711.13  4889.3  710.89  4916.5  711.92
  4959.0  712.66  4981.0  704.57  4983.0  704.07  4998.3  704.57  5009.7  711.05
  5019.7  715.08  5060.8  713.74  5100.0  712.86  5160.2  714.85  5198.7  714.16
  5220.4  715.01  5280.6  713.75  5451.2  714.01  5618.3  712.92  5709.8  714.86
  5847.1  715.09  6018.3  716.94  6086.9  718.54  6115.3  720.61  6205.9  723.81
#Mann=5,-1,0
  4412.9    0.05       0  4916.5    0.12       0  4981.0    0.07       0
  4998.3    0.12       0  5060.8    0.05       0
Bank Sta=4981,4998.3
Exp/Cntr=0.3,0.1

Type RM Length L Ch R = 1,16754,555,555,555
BEGIN DESCRIPTION:
Mapping XS fc340b97
END DESCRIPTION:
XS GIS Cut Line= 3
      2310888.12      7111322.82      2310272.47      7110399.65
      2310104.89      7110123.90
#Sta/Elev= 30
  4659.6  731.70  4668.0  732.45  4675.0  729.92  4683.0  728.80  4806.2  716.26
  4852.3  714.97  4905.4  709.40  4950.4  710.08  4956.4  707.73  4963.5  708.94
  4971.5  708.12  4977.5  704.69  4990.9  703.18  4992.9  702.68  5008.2  703.18
  5015.3  704.96  5022.5  707.02  5028.5  711.26  5035.6  713.77  5049.6  714.16
  5064.6  712.55  5130.7  711.22  5244.9  712.47  5347.0  711.62  5476.2  713.81
  5599.4  714.39  5635.4  715.56  5785.9  715.88  5981.7  718.28  6091.9  723.43
#Mann=5,-1,0
  4659.6    0.05       0  4852.3    0.12       0  4990.9    0.07       0
  5008.2    0.12       0  5015.3    0.05       0
Bank Sta=4990.9,5008.2
Exp/Cntr=0.3,0.1

Type RM Length L Ch R = 1,16199,758,758,758
BEGIN DESCRIPTION:
Mapping XS 98d48f69
END DESCRIPTION:
XS GIS Cut Line= 2
      2311364.50      7111029.22      2310343.57      7110191.88
#Sta/Elev= 30
  4392.6  733.45  4431.4  731.23  4445.8  725.98  4480.9  722.48  4503.2  718.75
  4544.8  715.93  4672.6  711.28  4829.0  709.93  4851.2  710.92  4857.7  712.17
  4872.8  710.24  4878.5  708.97  4886.4  710.43  4921.6  711.57  4935.9  708.68
  4979.0  708.63  4985.4  707.98  4999.8  702.42  5012.0  700.98  5014.0  700.48
  5029.3  700.98  5035.0  706.46  5049.3  711.22  5092.4  712.43  5127.5  711.88
  5149.8  709.94  5171.9  709.46  5248.8  709.59  5475.6  713.57  5713.0  716.13
#Mann=5,-1,0
  4392.6    0.05       0  4872.8    0.12       0  5012.0    0.07       0
  5029.3    0.12       0  5171.9    0.05       0
Bank Sta=5012,5029.3
Exp/Cntr=0.3,0.1

Type RM Length L Ch R = 1,15441,596,596,596
BEGIN DESCRIPTION:
Mapping XS 7cd4029d
END DESCRIPTION:
XS GIS Cut Line= 2
      2311525.66      7110598.08      2310517.81      7109653.64
#Sta/Elev= 30
  4197.0  719.35  4278.1  718.90  4285.4  717.95  4292.2  718.70  4299.5  715.71
  4306.4  716.13  4313.7  711.83  4320.6  711.15  4363.0  709.95  4419.7  709.71
  4483.2  707.21  4554.0  706.53  4667.4  707.54  4724.0  708.87  4787.5  708.00
  4858.3  705.49  4915.0  707.04  4950.2  706.07  4971.7  706.53  4978.5  705.82
  4983.9  697.60  4985.9  697.10  5001.4  697.60  5035.2  705.79  5049.3  710.49
  5063.5  708.91  5084.5  711.08  5169.5  710.80  5417.2  712.58  5578.2  715.63
#Mann=3,-1,0
  4197.0    0.05       0  4983.9   0.033       0  5001.4    0.05       0
Bank Sta=4983.9,5001.4
Exp/Cntr=0.3,0.1

Type RM Length L Ch R = 1,14845,358,358,358
BEGIN DESCRIPTION:
Mapping XS 19fd7996
END DESCRIPTION:
XS GIS Cut Line= 2
      2311591.78      7110542.48      2311091.28      7109000.47
#Sta/Elev= 30
  4368.8  719.33  4486.5  717.82  4491.7  714.34  4497.6  716.07  4518.4  716.66
  4523.7  711.92  4529.1  713.74  4550.1  714.08  4560.9  708.68  4644.8  706.21
  4834.0  705.51  4943.1  707.79  4949.8  705.13  4970.7  702.10  4981.7  698.18
  5002.2  697.02  5005.0  695.59  5007.0  695.09  5022.5  695.59  5023.2  700.33
  5033.8  704.38  5045.3  705.16  5086.3  708.33  5141.6  706.80  5422.8  706.78
  5811.8  708.93  5864.3  710.85  5919.3  716.15  5946.0  720.52  5990.0  723.01
#Mann=5,-1,0
  4368.8    0.05       0  4943.1    0.12       0  5005.0    0.07       0
  5022.5    0.12       0  5045.3    0.05       0
Bank Sta=5005,5022.5
Exp/Cntr=0.3,0.1

Type RM Length L Ch R = 1,14487,249,249,249
BEGIN DESCRIPTION:
Mapping XS 9d7a45a9
END DESCRIPTION:
XS GIS Cut Line= 2
      2311778.36      7110457.95      2311584.31      7109196.18
#Sta/Elev= 30
  4393.0  719.18  4431.4  719.07  4461.7  711.18  4482.0  710.72  4487.3  711.62
  4492.3  709.89  4502.2  709.85  4522.5  711.45  4542.7  711.77  4550.5  711.36
  4555.6  709.14  4583.2  708.50  4613.5  706.42  4942.9  703.48  4998.0  703.78
  5004.7  694.87  5006.7  694.37  5022.2  694.87  5050.0  698.97  5068.8  706.11
  5081.8  708.69  5089.0  707.38  5109.3  706.13  5250.9  705.04  5413.2  705.24
  5503.9  707.52  5602.9  714.75  5608.0  713.64  5645.5  715.66  5669.6  715.95
#Mann=5,-1,0
  4393.0    0.05       0  4942.9    0.12       0  5004.7    0.07       0
  5022.2    0.12       0  5050.0    0.05       0
Bank Sta=5004.7,5022.2
Exp/Cntr=0.3,0.1

Type RM Length L Ch R = 1,14238,796,796,796
BEGIN DESCRIPTION:
Mapping XS 20666229
END DESCRIPTION:
XS GIS Cut Line= 2
      2311991.49      7110545.06      2311856.14      7109310.76
#Sta/Elev= 30
  4351.3  731.26  4406.7  728.38  4446.9  719.43  4557.6  711.78  4597.8  707.19
  4842.9  706.64  4859.4  705.00  4869.4  702.59  4889.6  704.41  4919.7  702.11
  4949.9  703.78  4960.0  698.18  4967.7  698.87  4972.8  701.73  4980.1  701.44
  4990.2  696.24  5001.5  694.38  5003.5  693.88  5019.1  694.38  5020.3  696.82
  5040.5  703.27  5063.9  704.16  5080.7  702.55  5131.0  705.85  5150.0  704.18
  5185.0  704.44  5292.0  704.26  5362.4  705.48  5412.7  709.70  5593.0  712.92
#Mann=5,-1,0
  4351.3    0.05       0  4842.9    0.12       0  5001.5    0.07       0
  5019.1    0.12       0  5185.0    0.05       0
Bank Sta=5001.5,5019.1
Exp/Cntr=0.3,0.1

Type RM Length L Ch R = 1,13442,340,340,340
BEGIN DESCRIPTION:
Mapping XS 7140799e
END DESCRIPTION:
XS GIS Cut Line= 3
      2312691.37      7110188.93      2312585.71      7109720.29
      2312289.46      7108873.52
#Sta/Elev= 30
  4630.0  715.37  4707.4  709.98  4799.0  706.46  4813.4  706.64  4823.7  704.74
  4842.2  704.31  4847.3  703.19  4874.9  701.63  4946.7  700.55  4956.9  699.85
  4967.2  697.47  4977.0  692.47  4982.2  691.03  4988.8  690.86  4990.8  690.36
  5007.1  690.86  5008.2  693.11  5018.4  696.14  5025.1  697.19  5030.5  698.77
  5049.2  701.00  5096.8  699.82  5177.9  699.63  5184.9  700.62  5259.0  701.76
  5428.5  702.97  5492.1  704.54  5508.6  703.54  5627.5  705.09  6007.5  711.92
#Mann=5,-1,0
  4630.0    0.05       0  4988.8   0.033       0  5007.1    0.05       0
  5025.1    0.12       0  5096.8    0.05       0
Bank Sta=4988.8,5007.1
Exp/Cntr=0.3,0.1

Type RM Length L Ch R = 1,13102,545,545,545
BEGIN DESCRIPTION:
Morris Branch 15.0
END DESCRIPTION:
XS GIS Cut Line= 3
      2313129.01      7110110.02      2312929.00      7109760.00
      2312079.00      7108160.00
#Sta/Elev= 30
  4597.0  722.05  4685.6  713.73  4809.4  709.75  4846.8  705.82  4927.4  700.97
  4949.0  697.35  4954.8  697.44  4964.9  695.90  4977.1  697.21  4988.1  689.47
  4990.1  688.97  5006.4  689.47  5022.8  690.26  5030.3  698.86  5052.3  698.55
  5074.2  701.27  5102.1  699.64  5237.9  697.77  5376.3  700.18  5474.9  700.18
  5568.5  702.64  5584.8  701.81  5628.8  702.28  5859.2  706.65  5996.8  711.89
  6057.1  713.28  6199.6  719.56  6347.6  723.72  6589.6  732.54  6811.9  744.06
#Mann=3,-1,0
  4597.0    0.05       0  4988.1   0.033       0  5006.4    0.05       0
Bank Sta=4988.1,5006.4
Exp/Cntr=0.3,0.1

Type RM Length L Ch R = 1,12557,337,337,337
BEGIN DESCRIPTION:
Morris Branch 14.0
END DESCRIPTION:
XS GIS Cut Line= 3
      2313229.00      7110159.97      2313179.00      7109360.00
      2312029.02      7107760.03
#Sta/Elev= 30
  4202.9  726.05  4212.9  726.23  4222.9  723.84  4263.0  723.14  4383.2  714.25
  4533.5  709.84  4593.6  706.35  4613.7  703.75  4703.4  700.44  4761.5  699.43
  4804.0  701.25  4884.2  696.34  4909.2  696.47  4944.3  694.67  4954.3  692.91
  4955.2  688.61  4957.2  688.11  4973.5  688.61  4994.4  689.34  5001.9  698.12
  5007.5  698.12  5011.8  700.16  5139.9  696.56  5835.6  707.62  6223.5  725.54
  6573.4  744.03  6688.8  751.84  6795.6  757.32  6875.4  764.77  6974.8  771.24
#Mann=5,-1,0
  4202.9    0.05       0  4703.4    0.12       0  4909.2    0.05       0
  4955.2   0.033       0  4973.5    0.05       0
Bank Sta=4955.2,4973.5
Exp/Cntr=0.3,0.1

Type RM Length L Ch R = 1,12220,686,686,686
BEGIN DESCRIPTION:
Mapping XS 27e77fc8
END DESCRIPTION:
XS GIS Cut Line= 3
      2313495.26      7109797.21      2313401.93      7109158.07
      2313017.54      7108076.14
#Sta/Elev= 30
  4355.7  709.08  4571.1  702.30  4656.1  701.16  4716.7  698.43  4893.3  695.94
  4915.9  694.93  4933.3  696.20  4939.0  696.89  4959.2  694.72  4969.3  689.81
  4976.8  687.44  4978.8  686.94  4995.1  687.44  4998.1  689.29  5001.6  689.29
  5010.2  696.15  5020.4  697.11  5025.7  699.07  5031.4  699.64  5073.9  697.83
  5200.2  695.66  5385.3  697.91  5424.1  697.19  5893.9  705.49  5944.1  705.54
  6037.6  707.93  6050.2  709.42  6099.3  712.23  6113.9  715.05  6149.8  718.23
#Mann=5,-1,0
  4355.7    0.05       0  4893.3    0.12       0  4933.3    0.05       0
  4976.8   0.033       0  4995.1    0.05       0
Bank Sta=4976.8,4995.1
Exp/Cntr=0.3,0.1

Type RM Length L Ch R = 1,11534,561,561,561
BEGIN DESCRIPTION:
Mapping XS a164e123
END DESCRIPTION:
XS GIS Cut Line= 4
      2313826.55      7109602.28      2313695.58      7108914.45
      2313463.78      7108730.44      2313234.76      7108288.39
#Sta/Elev= 30
  4410.4  704.71  4473.1  703.59  4478.2  704.21  4494.2  703.92  4565.4  701.37
  4718.1  698.76  4779.2  696.26  4840.3  697.15  4860.6  698.93  4870.9  698.89
  4911.5  697.55  4931.9  694.08  4942.1  693.61  4952.2  692.11  4972.6  691.49
  4993.0  686.40  5003.1  686.08  5006.1  683.35  5008.1  682.85  5024.5  683.35
  5033.7  694.60  5043.9  698.20  5054.0  698.63  5067.4  697.50  5196.0  694.14
  5338.6  696.69  5396.4  696.36  5580.8  698.72  5602.9  700.93  5904.4  702.26
#Mann=4,-1,0
  4410.4    0.05       0  4870.9    0.12       0  5006.1    0.07       0
  5024.5    0.05       0
Bank Sta=5006.1,5024.5
Exp/Cntr=0.3,0.1

Type RM Length L Ch R = 1,10973,520,520,520
BEGIN DESCRIPTION:
Morris Branch 11.0
END DESCRIPTION:
XS GIS Cut Line= 3
      2314078.99      7109660.05      2314179.00      7108860.00
      2313678.99      7108059.98
#Sta/Elev= 30
  4194.2  712.72  4232.0  709.91  4496.6  698.72  4788.8  693.71  4869.5  694.99
  4919.9  692.94  4957.6  694.77  4967.3  693.88  4990.4  692.82  4998.0  687.18
  5003.4  687.18  5008.1  682.07  5020.1  681.84  5022.1  681.34  5038.6  681.84
  5044.7  691.04  5050.6  690.94  5065.9  694.50  5078.1  695.65  5094.8  696.76
  5102.5  695.13  5327.7  690.10  5413.2  693.10  5625.5  696.16  5653.2  697.47
  5726.3  707.02  5784.1  709.89  5820.6  713.66  5878.4  716.71  5943.9  722.03
#Mann=5,-1,0
  4194.2    0.05       0  4967.3    0.12       0  5020.1    0.07       0
  5038.6    0.12       0  5078.1    0.05       0
Bank Sta=5020.1,5038.6
Exp/Cntr=0.3,0.1

Type RM Length L Ch R = 1,10453,682,682,682
BEGIN DESCRIPTION:
MAPPING XS 96962
END DESCRIPTION:
XS GIS Cut Line= 2
      2314839.34      7109121.74      2314161.69      7107938.67
#Sta/Elev= 30
  4618.2  703.24  4700.9  702.20  4713.8  699.54  4771.0  697.03  4804.4  693.12
  4810.2  690.79  4816.1  690.21  4885.0  689.17  4890.8  687.97  4906.6  687.93
  4912.3  686.39  4928.2  687.05  4933.9  683.07  4942.9  683.72  4955.5  681.21
  4977.9  680.64  4979.9  680.14  4996.5  680.64  5000.5  682.86  5008.7  684.03
  5014.5  691.83  5023.5  693.13  5145.8  692.30  5403.8  692.08  5433.2  690.66
  5454.8  687.16  5470.6  689.23  5556.9  691.85  5820.2  692.53  5981.6  694.97
#Mann=5,-1,0
  4618.2    0.05       0  4771.0    0.12       0  4977.9    0.07       0
  4996.5    0.12       0  5145.8    0.05       0
Bank Sta=4977.9,4996.5
Exp/Cntr=0.3,0.1

Type RM Length L Ch R = 1,9771,605,605,605
BEGIN DESCRIPTION:
Mapping XS b90dab14
END DESCRIPTION:
XS GIS Cut Line= 2
      2315052.06      7108957.26      2315074.16      7107447.62
#Sta/Elev= 30
  4471.7  702.83  4649.0  699.84  4779.0  691.53  4849.0  688.65  4905.2  689.68
  4929.0  689.78  4959.0  686.86  4979.0  682.49  4989.0  681.57  4999.0  679.41
  4999.7  678.11  5001.7  677.61  5018.3  678.11  5019.0  679.39  5029.0  678.60
  5039.0  679.89  5049.0  684.81  5069.0  688.77  5089.0  690.22  5129.0  688.67
  5186.4  688.92  5359.1  689.81  5439.1  688.30  5499.1  689.40  5629.1  688.81
  5799.1  692.11  5819.1  693.61  5889.1  709.21  5919.1  714.34  5981.5  717.88
#Mann=5,-1,0
  4471.7    0.05       0  4905.2    0.12       0  4999.7    0.07       0
  5018.3    0.12       0  5186.4    0.05       0
Bank Sta=4999.7,5018.3
Exp/Cntr=0.3,0.1

Type RM Length L Ch R = 1,9166,695,695,695
BEGIN DESCRIPTION:
Mapping XS f97d95a8
END DESCRIPTION:
XS GIS Cut Line= 2
      2315558.41      7108997.30      2315514.82      7107639.30
#Sta/Elev= 30
  4712.5  698.70  4852.5  695.23  4899.9  695.56  4919.9  694.59  4929.9  693.81
  4939.9  691.14  4959.9  683.49  4989.9  679.50  4999.9  677.35  5010.0  677.35
  5010.7  676.82  5012.7  676.32  5029.3  676.82  5040.0  685.59  5050.0  687.66
  5060.0  688.66  5080.0  688.76  5100.0  689.90  5110.0  690.02  5120.0  688.79
  5150.0  688.38  5230.1  688.77  5410.2  688.08  5540.2  686.12  5660.3  686.65
  5720.3  686.23  5880.4  689.62  6000.5  693.06  6030.5  694.60  6071.2  698.96
#Mann=3,-1,0
  4712.5    0.05       0  5010.7   0.033       0  5029.3    0.05       0
Bank Sta=5010.7,5029.3
Exp/Cntr=0.3,0.1

Type RM Length L Ch R = 1,8471,672,672,672
BEGIN DESCRIPTION:
Mapping XS 0016a320
END DESCRIPTION:
XS GIS Cut Line= 2
      2316247.37      7108770.38      2315684.03      7107315.00
#Sta/Elev= 30
  4668.6  699.27  4754.8  697.69  4785.2  698.21  4797.7  696.32  4899.6  690.96
  4915.6  688.23  4929.5  683.88  4947.8  682.83  4959.4  680.93  4981.4  674.38
  4983.4  673.88  5000.0  674.38  5001.4  676.20  5008.6  680.30  5013.9  682.11
  5022.9  682.34  5055.0  687.02  5286.5  684.32  5473.2  685.46  5559.0  684.03
  5580.5  682.23  5601.9  684.85  5634.1  685.71  5787.8  687.14  5827.1  685.68
  5902.2  689.71  6030.4  691.74  6095.7  694.51  6180.9  701.90  6229.2  704.41
#Mann=3,-1,0
  4668.6    0.05       0  4981.4   0.035       0  5000.0    0.05       0
Bank Sta=4981.4,5000
Exp/Cntr=0.3,0.1

Type RM Length L Ch R = 1,7799,301,301,301
BEGIN DESCRIPTION:
Mapping XS c721766e
END DESCRIPTION:
XS GIS Cut Line= 2
      2316743.81      7108431.06      2316126.40      7107104.72
#Sta/Elev= 30
  4558.7  693.68  4744.8  689.67  4875.8  684.34  4968.0  679.38  4990.2  673.70
  4998.2  673.57  5000.2  673.07  5016.8  673.57  5030.4  678.04  5035.9  683.72
  5089.3  682.51  5133.4  684.25  5150.3  681.56  5155.8  682.95  5166.5  676.84
  5173.2  679.24  5178.7  676.34  5196.1  678.37  5201.6  676.17  5211.2  677.11
  5219.0  677.03  5247.3  682.67  5287.6  677.33  5293.1  678.05  5298.9  683.60
  5596.0  684.26  5872.5  688.05  5932.9  694.80  5978.6  703.80  6021.7  709.66
#Mann=5,-1,0
  4558.7    0.05       0  4875.8    0.12       0  4998.2    0.07       0
  5016.8    0.12       0  5211.2    0.05       0
Bank Sta=4998.2,5016.8
Exp/Cntr=0.3,0.1

Type RM Length L Ch R = 1,7498,130,130,130
BEGIN DESCRIPTION:
Mapping XS b5d6c2db
END DESCRIPTION:
XS GIS Cut Line= 2
      2316830.23      7108600.82      2316729.56      7106884.88
#Sta/Elev= 30
  4308.1  697.42  4459.2  695.45  4469.2  694.23  4509.3  693.22  4789.8  688.47
  4839.8  683.20  4899.9  682.98  4920.0  682.00  4925.9  680.50  4940.0  680.12
  4950.0  678.49  4960.0  678.90  4970.1  676.40  4980.1  675.47  4980.7  674.22
  4982.7  673.72  4999.5  674.22  5010.1  674.24  5030.2  680.71  5070.2  681.49
  5090.3  683.56  5170.4  682.34  5437.4  683.39  5631.2  682.77  5791.5  683.85
  5841.6  686.55  5901.7  693.55  5931.7  702.66  5949.0  706.32  6027.0  713.04
#Mann=3,-1,0
  4308.1    0.05       0  4980.7   0.033       0  4999.5    0.05       0
Bank Sta=4980.7,4999.5
Exp/Cntr=0.3,0.1

Type RM Length L Ch R = 1,7368,414,414,414
BEGIN DESCRIPTION:
Mapping XS 383e5dc5
END DESCRIPTION:
XS GIS Cut Line= 2
      2316949.50      7108602.19      2316852.93      7106850.55
#Sta/Elev= 30
  4276.3  697.50  4629.0  689.61  4689.1  689.10  4741.9  690.35  4789.3  690.01
  4869.4  684.65  4959.5  682.47  4979.6  674.46  4990.2  673.93  4992.2  673.43
  5009.0  673.93  5009.6  675.68  5019.6  675.68  5039.6  678.85  5049.7  678.85
  5069.7  681.05  5119.8  682.63  5199.9  682.57  5239.9  680.53  5310.1  682.42
  5357.8  682.58  5363.1  682.42  5651.7  682.04  5740.7  683.94  5820.8  687.88
  5901.0  693.54  5931.0  698.97  5951.0  701.22  5981.1  706.92  6030.6  711.56
#Mann=5,-1,0
  4276.3    0.05       0  4990.2    0.04       0  5009.0    0.05       0
  5357.8    0.12       0  5363.1    0.05       0
Bank Sta=4990.2,5009
Exp/Cntr=0.3,0.1

Type RM Length L Ch R = 1,6954,369,369,369
BEGIN DESCRIPTION:
Mapping XS 363555eb
END DESCRIPTION:
XS GIS Cut Line= 3
      2317172.33      7108648.95      2317277.39      7107824.14
      2317333.53      7106676.79
#Sta/Elev= 30
  4104.2  698.24  4365.2  689.69  4445.9  690.37  4556.8  682.16  4655.6  680.93
  4728.2  681.24  4758.4  678.18  4849.1  680.38  4940.3  679.36  4990.5  672.44
  4992.5  671.94  5009.3  672.44  5009.9  675.08  5019.9  677.16  5060.0  682.69
  5090.0  680.32  5230.2  681.70  5280.3  677.28  5361.0  680.49  5380.3  679.21
  5433.5  682.67  5530.5  687.50  5661.3  688.55  5780.8  692.64  5880.9  702.46
  5901.0  702.29  5921.0  706.32  5941.0  706.26  6001.1  713.44  6084.4  718.81
#Mann=7,-1,0
  4104.2    0.05       0  4655.6    0.12       0  4990.5    0.07       0
  5009.3    0.12       0  5361.0    0.05       0  5433.5    0.12       0
  5661.3    0.05       0
Bank Sta=4990.5,5009.3
Exp/Cntr=0.3,0.1

Type RM Length L Ch R = 1,6585,250,250,250
BEGIN DESCRIPTION:
Mapping XS ad51f47e
END DESCRIPTION:
XS GIS Cut Line= 3
      2317360.27      7108640.62      2317577.63      7107936.48
      2317539.17      7106653.98
#Sta/Elev= 30
  4279.5  696.60  4429.8  686.20  4462.5  682.30  4500.4  680.87  4565.7  679.32
  4892.9  679.60  4950.6  679.46  4960.4  677.69  4967.9  675.17  4991.8  675.02
  5000.6  673.08  5002.6  670.62  5004.6  670.12  5021.4  670.62  5022.9  671.92
  5072.9  673.53  5092.9  679.34  5143.0  679.44  5183.0  680.97  5243.0  679.74
  5663.2  679.43  5763.2  680.65  5903.3  684.64  5923.3  686.38  5953.3  686.93
  6023.4  690.95  6073.4  695.46  6123.4  703.24  6153.4  703.48  6299.5  717.42
#Mann=5,-1,0
  4279.5    0.05       0  4892.9    0.12       0  4950.6    0.05       0
  5002.6   0.033       0  5021.4    0.05       0
Bank Sta=5002.6,5021.4
Exp/Cntr=0.3,0.1
