HEC-RAS study Oliver Creek.prj: Oliver Creek Base Level Engineering

--- Oliver Creek.g01 (geometry) --- (continued)

Type RM Length L Ch R = 1,105753,456,456,456
BEGIN DESCRIPTION:
Oliver Creek 133.0
END DESCRIPTION:
XS GIS Cut Line= 3
      2265090.40      7113084.31      2264995.31      7112641.92
      2264606.63      7112144.82
#Sta/Elev= 30
  4566.5  902.32  4663.0  901.50  4739.7  899.35  4806.2  898.41  4918.7  894.69
  4932.0  895.32  4957.8  887.70  4969.8  885.55  4976.3  883.65  4981.4  884.23
  5010.7  872.91  5013.5  868.27  5014.7  867.77  5021.4  868.27  5024.4  869.84
  5032.6  877.82  5053.4  889.23  5074.2  893.78  5082.3  893.00  5111.4  892.79
  5351.8  895.37  5402.2  895.12  5502.8  897.05  5567.0  901.77  5594.2  907.60
  5608.6  912.69  5616.7  916.77  5623.1  917.65  5637.6  921.61  5650.0  923.07
#Mann=5,-1,0
  4566.5    0.05       0  4957.8    0.12       0  5013.5    0.07       0
  5021.4    0.12       0  5111.4    0.05       0
Bank Sta=5013.5,5021.4
Exp/Cntr=0.3,0.1

Type RM Length L Ch R = 1,105297,366,366,366
BEGIN DESCRIPTION:
Mapping XS a8d7375a
END DESCRIPTION:
XS GIS Cut Line= 2
      2265289.48      7112450.36      2264938.57      7111997.63
#Sta/Elev= 30
  4785.0  891.30  4874.0  890.40  4906.9  890.26  4921.4  889.30  4927.7  889.60
  4949.9  888.84  4956.7  886.36  4963.0  886.40  4977.5  881.27  4985.7  879.58
  5000.2  874.17  5006.5  869.40  5017.0  866.32  5018.2  865.82  5023.7  865.82
  5024.9  866.32  5027.3  868.96  5035.5  873.89  5041.8  882.31  5050.0  885.70
  5056.3  889.82  5077.1  892.37  5091.6  893.20  5106.1  892.77  5141.4  894.42
  5183.9  897.52  5234.6  901.09  5255.5  901.44  5342.2  908.20  5357.8  908.80
#Mann=5,-1,0
  4785.0    0.05       0  4874.0    0.12       0  5017.0    0.07       0
  5024.9    0.12       0  5183.9    0.05       0
Bank Sta=5017,5024.9
Exp/Cntr=0.3,0.1

Type RM Length L Ch R = 1,104931,530,530,530
BEGIN DESCRIPTION:
Mapping XS 8384ae11
END DESCRIPTION:
XS GIS Cut Line= 2
      2265476.59      7112533.81      2265481.58      7111994.73
#Sta/Elev= 30
  4731.0  890.29  4804.8  889.60  4834.8  889.67  4894.8  889.23  4904.8  889.28
  4914.8  889.76  4924.8  889.47  4934.8  886.77  4944.8  880.57  4946.2  878.96
  4954.8  869.05  4960.7  864.08  4961.9  863.58  4967.7  863.58  4969.0  864.08
  4974.8  864.18  4994.8  876.56  5004.8  881.39  5014.8  884.14  5034.8  886.69
  5044.8  888.82  5064.8  890.29  5074.8  889.96  5094.8  890.95  5104.8  891.73
  5114.8  891.63  5134.8  892.90  5210.9  896.33  5264.8  899.36  5270.1  899.87
#Mann=5,-1,0
  4731.0    0.05       0  4946.2    0.12       0  4960.7    0.07       0
  4969.0    0.12       0  5210.9    0.05       0
Bank Sta=4960.7,4969
Exp/Cntr=0.3,0.1

Type RM Length L Ch R = 1,104401,574,574,574
BEGIN DESCRIPTION:
Oliver Creek 131.0
END DESCRIPTION:
XS GIS Cut Line= 3
      2265749.05      7112521.07      2265929.56      7112107.61
      2265920.43      7111714.26
#Sta/Elev= 30
  4550.6  886.79  4740.3  885.25  4816.0  885.46  4873.6  883.71  4886.2  883.17
  4900.9  883.94  4909.6  881.38  4915.1  882.14  4922.8  878.91  4933.0  876.82
  4938.5  877.80  4944.6  874.63  4961.9  875.32  4977.3  874.74  4985.3  873.00
  4990.8  873.63  4997.7  871.61  5001.8  871.61  5009.4  862.13  5015.2  861.86
  5016.4  861.36  5023.5  861.86  5039.4  873.54  5059.4  882.90  5069.4  886.01
  5081.9  886.35  5109.4  886.41  5229.4  889.01  5389.5  896.83  5395.2  897.84
#Mann=5,-1,0
  4550.6    0.05       0  4873.6    0.12       0  5015.2    0.07       0
  5023.5    0.12       0  5081.9    0.05       0
Bank Sta=5015.2,5023.5
Exp/Cntr=0.3,0.1

Type RM Length L Ch R = 1,103827,380,380,380
BEGIN DESCRIPTION:
Oliver Creek 130.0
END DESCRIPTION:
XS GIS Cut Line= 3
      2266560.64      7112506.99      2266344.72      7112310.72
      2265929.02      7111710.03
#Sta/Elev= 30
  4708.2  893.99  4770.9  893.64  4785.1  891.35  4905.4  886.45  4919.6  885.17
  4933.8  882.08  4940.5  882.22  4952.4  878.23  4968.9  870.65  4976.4  869.75
  4983.1  863.58  4990.5  860.34  4990.9  857.46  4992.5  856.96  5002.8  857.46
  5012.9  864.56  5019.0  871.08  5025.2  872.39  5061.7  874.99  5090.6  879.68
  5105.5  880.12  5126.4  882.59  5141.3  882.10  5198.5  883.42  5371.0  885.01
  5385.9  884.16  5421.7  884.27  5529.2  885.94  5594.7  888.06  5730.5  897.09
#Mann=5,-1,0
  4708.2    0.05       0  4952.4    0.12       0  4990.9    0.07       0
  5002.8    0.12       0  5198.5    0.05       0
Bank Sta=4990.9,5002.8
Exp/Cntr=0.3,0.1

Type RM Length L Ch R = 1,103447,426,426,426
BEGIN DESCRIPTION:
Oliver Creek 129.0
END DESCRIPTION:
XS GIS Cut Line= 3
      2266704.96      7112310.55      2266418.04      7111970.40
      2265992.71      7111582.57
#Sta/Elev= 30
  4555.0  891.86  4765.0  883.80  4788.9  880.42  4864.9  876.34  4885.8  871.81
  4893.5  874.89  4900.1  873.51  4963.8  870.47  4971.5  869.67  4978.1  864.08
  4991.0  859.81  4992.7  859.31  5002.9  859.81  5013.5  862.51  5020.9  875.19
  5035.1  880.90  5070.3  883.46  5091.9  882.30  5112.8  878.73  5120.3  878.73
  5127.0  878.52  5148.0  882.38  5204.7  881.87  5233.1  883.74  5325.0  884.65
  5431.7  889.99  5502.0  891.58  5558.7  895.28  5572.9  897.87  5575.6  899.60
#Mann=5,-1,0
  4555.0    0.05       0  4788.9    0.12       0  4991.0    0.07       0
  5002.9    0.12       0  5120.3    0.05       0
Bank Sta=4991,5002.9
Exp/Cntr=0.3,0.1

Type RM Length L Ch R = 1,103021,462,462,462
BEGIN DESCRIPTION:
Oliver Creek 128.0
END DESCRIPTION:
XS GIS Cut Line= 3
      2266920.24      7112199.44      2266723.81      7111709.56
      2266379.23      7111254.13
#Sta/Elev= 30
  4472.2  888.59  4736.3  882.32  4762.8  879.47  4794.8  877.48  4811.2  877.61
  4816.6  875.31  4835.4  873.29  4840.8  870.86  4859.5  870.48  4870.4  868.74
  4902.6  867.42  4978.0  868.83  4988.7  866.31  4993.7  858.37  4995.4  857.87
  5005.7  858.37  5011.0  859.83  5017.3  858.89  5024.5  863.23  5031.8  875.10
  5046.4  878.51  5060.9  880.32  5067.2  879.38  5088.5  880.79  5267.0  882.71
  5396.0  886.21  5516.7  893.58  5524.9  895.09  5566.6  897.00  5571.1  898.24
#Mann=5,-1,0
  4472.2    0.05       0  4736.3    0.12       0  4993.7    0.07       0
  5005.7    0.12       0  5088.5    0.05       0
Bank Sta=4993.7,5005.7
Exp/Cntr=0.3,0.1

Type RM Length L Ch R = 1,102559,270,270,270
BEGIN DESCRIPTION:
Oliver Creek 127.0
END DESCRIPTION:
XS GIS Cut Line= 3
      2267307.38      7111923.38      2267125.45      7111551.50
      2266795.26      7111077.95
#Sta/Elev= 30
  4586.0  888.12  4834.7  882.40  4856.9  881.39  4870.2  879.71  4879.2  880.62
  4887.2  880.30  4904.4  878.54  4915.2  878.65  4937.7  872.71  4946.0  869.62
  4954.7  871.14  4960.2  867.92  4968.3  869.98  4977.2  869.47  4990.5  859.00
  4998.1  855.83  4999.2  854.64  5000.9  854.14  5011.2  854.64  5014.0  859.38
  5020.1  861.57  5026.2  868.21  5049.7  868.88  5099.4  876.06  5121.3  877.71
  5143.8  877.45  5184.7  878.66  5365.6  879.88  5493.8  884.00  5577.3  889.53
#Mann=5,-1,0
  4586.0    0.05       0  4904.4    0.12       0  4999.2    0.07       0
  5011.2    0.12       0  5143.8    0.05       0
Bank Sta=4999.2,5011.2
Exp/Cntr=0.3,0.1

Type RM Length L Ch R = 1,102289,418,418,418
BEGIN DESCRIPTION:
Mapping XS f77ec92c
END DESCRIPTION:
XS GIS Cut Line= 3
      2267472.98      7111688.74      2267236.58      7111242.51
      2267068.76      7111309.04
#Sta/Elev= 30
  4613.3  888.15  4718.6  887.12  4757.0  884.69  4806.6  882.47  4838.2  880.42
  4850.6  878.90  4860.8  876.58  4867.0  876.34  4872.6  873.13  4883.3  873.23
  4889.0  869.82  4940.0  865.76  4955.0  865.60  4962.7  863.95  4971.0  854.34
  4972.6  853.84  4981.3  853.84  4983.0  854.34  4985.3  854.53  4993.3  857.26
  4999.0  861.38  5021.0  867.66  5030.6  867.96  5053.2  873.46  5071.2  874.64
  5109.8  877.10  5177.1  876.86  5206.8  877.53  5212.5  877.07  5298.8  877.76
#Mann=5,-1,0
  4613.3    0.05       0  4872.6    0.12       0  4971.0    0.07       0
  4983.0    0.12       0  5071.2    0.05       0
Bank Sta=4971,4983
Exp/Cntr=0.3,0.1

Type RM Length L Ch R = 1,101871,223,223,223
BEGIN DESCRIPTION:
Mapping XS c5567c04
END DESCRIPTION:
XS GIS Cut Line= 2
      2267736.26      7111465.14      2267444.75      7110583.69
#Sta/Elev= 30
  4625.5  879.66  4766.7  876.91  4851.2  876.01  4873.2  871.41  4904.8  867.23
  4983.4  864.29  4989.0  862.86  4999.6  864.24  5015.1  861.59  5020.6  857.64
  5031.2  854.41  5040.8  853.39  5042.5  852.89  5052.9  853.39  5062.8  866.06
  5083.8  875.29  5147.3  876.01  5240.1  882.65  5274.2  885.04  5300.6  889.43
  5305.9  888.60  5332.3  894.93  5337.6  893.29  5364.1  903.71  5369.3  903.12
  5395.8  908.46  5432.8  909.63  5522.7  909.28  5536.7  910.41  5553.9  909.52
#Mann=5,-1,0
  4625.5    0.05       0  4766.7    0.12       0  5040.8    0.07       0
  5052.9    0.12       0  5240.1    0.05       0
Bank Sta=5040.8,5052.9
Exp/Cntr=0.3,0.1

Type RM Length L Ch R = 1,101648,247,247,247
BEGIN DESCRIPTION:
Oliver Creek 125.0
END DESCRIPTION:
XS GIS Cut Line= 3
      2267807.40      7111527.54      2267826.67      7111065.75
      2267826.49      7110820.95
#Sta/Elev= 30
  4537.8  880.06  4585.4  879.30  4685.5  876.04  4853.3  874.48  4895.7  875.17
  4915.7  873.17  4933.4  866.99  4938.4  868.01  4945.7  864.71  4955.7  863.93
  4975.7  864.22  4995.4  853.30  4999.7  852.80  5001.4  852.30  5010.1  852.30
  5011.8  852.80  5015.7  853.57  5025.7  860.63  5035.7  865.94  5055.7  866.16
  5065.7  867.70  5075.7  870.29  5105.7  879.86  5125.7  883.38  5135.7  885.74
  5155.7  891.39  5160.9  893.68  5175.7  899.00  5195.7  903.63  5244.8  905.23
#Mann=5,-1,0
  4537.8    0.05       0  4853.3    0.12       0  4999.7    0.07       0
  5011.8    0.12       0  5160.9    0.05       0
Bank Sta=4999.7,5011.8
Exp/Cntr=0.3,0.1

Type RM Length L Ch R = 1,101401,210,210,210
BEGIN DESCRIPTION:
Mapping XS a88cac1a
END DESCRIPTION:
XS GIS Cut Line= 2
      2268055.79      7111348.20      2268085.74      7110839.08
#Sta/Elev= 30
  4711.3  874.45  4729.5  874.06  4769.6  870.86  4847.9  872.81  4852.9  872.50
  4859.8  873.43  4876.9  873.11  4899.8  872.30  4919.9  873.32  4929.9  870.37
  4949.9  868.18  4959.9  866.35  4969.9  866.51  4980.0  864.72  5000.0  863.86
  5018.2  859.03  5023.2  858.71  5030.0  856.17  5034.0  853.41  5035.7  852.91
  5044.4  852.91  5046.1  853.41  5050.1  856.91  5060.1  867.56  5070.1  876.34
  5080.1  880.84  5090.1  884.56  5100.2  886.23  5157.3  887.86  5221.3  887.62
#Mann=5,-1,0
  4711.3    0.05       0  4876.9    0.12       0  5034.0    0.07       0
  5046.1    0.12       0  5157.3    0.05       0
Bank Sta=5034,5046.1
Exp/Cntr=0.3,0.1

Type RM Length L Ch R = 1,101191,379,379,379
BEGIN DESCRIPTION:
Mapping XS c165ae70
END DESCRIPTION:
XS GIS Cut Line= 3
      2268182.06      7111316.73      2268281.61      7111208.65
      2268284.89      7110857.20
#Sta/Elev= 30
  4704.0  871.95  4706.6  872.44  4713.4  870.94  4720.8  871.50  4727.6  870.54
  4733.2  870.88  4741.8  869.68  4763.3  871.37  4812.6  872.34  4899.6  871.24
  4909.6  869.54  4919.6  865.11  4929.6  863.25  4949.6  860.67  4959.6  860.56
  4969.6  858.27  4979.6  853.84  4993.5  851.19  4995.2  850.69  5005.6  851.19
  5017.8  856.05  5019.6  856.71  5029.6  866.23  5039.6  870.52  5049.6  870.45
  5069.6  872.00  5089.6  871.10  5119.6  871.63  5179.6  874.61  5202.4  877.06
#Mann=5,-1,0
  4704.0    0.05       0  4733.2    0.12       0  4993.5    0.07       0
  5005.6    0.12       0  5017.8    0.05       0
Bank Sta=4993.5,5005.6
Exp/Cntr=0.3,0.1

Type RM Length L Ch R = 1,100812,393,393,393
BEGIN DESCRIPTION:
Oliver Creek 123.6
END DESCRIPTION:
XS GIS Cut Line= 3
      2268674.59      7111420.81      2268613.94      7111009.86
      2268505.32      7110629.15
#Sta/Elev= 30
  4584.6  877.10  4777.5  870.18  4807.8  870.93  4898.8  870.24  4919.0  867.67
  4932.6  864.73  4949.3  863.80  4969.5  861.31  4989.8  853.49  4993.7  850.55
  4995.4  850.05  5005.9  850.55  5010.3  851.32  5020.7  856.29  5036.2  860.73
  5051.8  858.86  5062.2  858.57  5074.0  859.62  5083.0  862.13  5103.8  865.75
  5109.1  869.67  5124.6  870.86  5260.0  872.91  5288.6  872.46  5343.0  876.95
  5361.6  880.50  5366.6  880.27  5384.6  883.80  5392.9  887.18  5395.9  887.18
#Mann=5,-1,0
  4584.6    0.05       0  4993.7   0.033       0  5005.9    0.05       0
  5074.0    0.12       0  5361.6    0.05       0
Bank Sta=4993.7,5005.9
Exp/Cntr=0.3,0.1

Type RM Length L Ch R = 1,100419,369,369,369
BEGIN DESCRIPTION:
Oliver Creek 123.4
END DESCRIPTION:
XS GIS Cut Line= 3
      2269006.67      7111092.85      2268959.05      7110880.12
      2268828.44      7110514.76
#Sta/Elev= 30
  4782.0  874.31  4842.5  872.74  4884.0  871.90  4889.1  870.31  4918.1  868.43
  4927.4  865.99  4932.5  865.74  4938.6  862.39  4948.9  859.68  4969.4  858.02
  4975.9  858.99  4981.0  858.30  4997.5  850.91  5002.7  850.91  5004.1  848.72
  5005.8  848.22  5016.3  848.72  5021.4  853.56  5032.0  859.49  5046.3  863.35
  5107.9  866.51  5133.3  865.00  5170.0  867.73  5194.9  867.67  5284.0  876.14
  5307.4  879.07  5318.7  881.84  5329.3  882.81  5350.6  886.65  5388.0  889.14
#Mann=5,-1,0
  4782.0    0.05       0  4842.5    0.12       0  5004.1    0.07       0
  5016.3    0.12       0  5284.0    0.05       0
Bank Sta=5004.1,5016.3
Exp/Cntr=0.3,0.1

Type RM Length L Ch R = 1,100050,279,279,279
BEGIN DESCRIPTION:
Oliver Creek 123.2
END DESCRIPTION:
XS GIS Cut Line= 3
      2269105.24      7111003.49      2269305.43      7110805.91
      2269034.98      7110339.52
#Sta/Elev= 30
  4592.5  871.00  4661.3  869.62  4675.4  870.60  4746.1  867.61  4802.7  867.51
  4897.2  866.03  4903.7  861.28  4913.0  856.89  4928.4  847.92  4930.1  847.42
  4940.6  847.92  4956.0  850.13  4961.8  852.06  4993.3  859.09  5030.6  858.64
  5052.1  857.03  5095.2  857.62  5138.2  859.86  5154.0  859.60  5169.6  862.65
  5175.5  865.41  5197.0  866.49  5234.3  870.20  5240.1  869.73  5255.8  870.31
  5351.0  875.96  5379.2  878.28  5395.0  882.29  5409.7  888.57  5412.9  888.57
#Mann=4,-1,0
  4592.5    0.12       0  4928.4    0.07       0  4940.6    0.12       0
  5351.0    0.05       0
Bank Sta=4928.4,4940.6
Exp/Cntr=0.3,0.1

Type RM Length L Ch R = 1,99771,331,331,331
BEGIN DESCRIPTION:
Mapping XS 960dd665
END DESCRIPTION:
XS GIS Cut Line= 3
      2269729.58      7110960.65      2269467.75      7110541.39
      2269266.48      7110256.15
#Sta/Elev= 30
  4467.8  871.55  4607.3  867.00  4689.0  865.89  4774.8  864.82  4796.0  865.97
  4904.8  862.71  4917.5  861.57  4932.8  857.32  4948.2  855.62  4960.0  848.04
  4965.3  848.04  4969.3  854.01  4976.0  855.15  4984.1  854.29  4990.2  855.74
  4998.8  851.10  5005.0  854.02  5012.8  848.48  5034.3  846.71  5036.1  846.21
  5047.0  846.71  5049.3  850.97  5055.5  850.60  5061.7  857.98  5070.3  864.18
  5076.4  865.08  5206.9  870.30  5227.9  873.68  5257.4  873.07  5311.2  875.95
#Mann=4,-1,0
  4467.8    0.05       0  4689.0    0.12       0  5034.3    0.07       0
  5047.0    0.12       0
Bank Sta=5034.3,5047
Exp/Cntr=0.3,0.1

Type RM Length L Ch R = 1,99440,479,479,479
BEGIN DESCRIPTION:
Oliver Creek 123.0
END DESCRIPTION:
XS GIS Cut Line= 3
      2270063.81      7110888.21      2269639.36      7110319.61
      2269287.73      7110010.56
#Sta/Elev= 30
  4240.8  871.75  4321.9  868.28  4421.9  866.12  4645.0  863.33  4692.9  863.27
  4707.5  861.83  4786.8  860.29  4800.1  860.98  4822.2  859.08  4857.6  858.38
  4922.3  858.68  4953.8  857.81  4978.3  855.29  4985.9  851.24  4992.5  851.29
  5000.1  847.96  5006.8  848.67  5014.6  846.81  5016.4  846.31  5027.3  846.81
  5042.8  856.32  5049.5  857.75  5057.0  862.49  5070.7  866.18  5113.0  870.55
  5130.6  870.69  5212.6  877.19  5262.0  882.20  5347.4  895.21  5418.5  897.31
#Mann=5,-1,0
  4240.8    0.05       0  4645.0    0.12       0  5014.6    0.07       0
  5027.3    0.12       0  5130.6    0.05       0
Bank Sta=5014.6,5027.3
Exp/Cntr=0.3,0.1

Type RM Length L Ch R = 1,98961,366,366,366
BEGIN DESCRIPTION:
Oliver Creek 122.0
END DESCRIPTION:
XS GIS Cut Line= 4
      2270082.02      7110854.31      2269957.03      7110388.20
      2269954.21      7110109.89      2269904.95      7109765.80
#Sta/Elev= 30
  4239.1  870.95  4384.6  865.64  4554.2  863.37  4574.3  861.80  4584.4  862.64
  4605.9  861.21  4619.5  861.93  4654.3  859.26  4668.0  859.83  4699.5  856.38
  4718.2  851.54  4859.9  854.58  4879.9  854.66  4899.9  853.04  4919.9  854.80
  4949.9  855.21  4969.9  853.15  4989.9  846.68  5003.6  844.61  5005.4  844.11
  5016.3  844.61  5020.1  849.07  5030.2  857.41  5040.3  862.41  5084.8  867.94
  5191.8  878.05  5215.1  884.59  5242.3  889.04  5292.8  891.40  5347.6  892.18
#Mann=5,-1,0
  4239.1    0.05       0  4584.4    0.12       0  5003.6    0.07       0
  5016.3    0.12       0  5084.8    0.05       0
Bank Sta=5003.6,5016.3
Exp/Cntr=0.3,0.1

Type RM Length L Ch R = 1,98595,801,801,801
BEGIN DESCRIPTION:
Oliver Creek 121.0
END DESCRIPTION:
XS GIS Cut Line= 3
      2270279.01      7110810.03      2270149.23      7110260.65
      2270037.77      7109797.06
#Sta/Elev= 30
  4435.5  874.83  4599.9  865.14  4733.5  861.41  4792.5  861.54  4826.0  859.38
  4856.8  853.94  4867.1  853.25  4908.2  855.44  4928.7  851.73  4934.8  848.84
  4977.1  845.76  4991.4  843.24  4993.2  842.74  5004.1  843.24  5019.2  845.82
  5026.4  851.80  5031.5  853.66  5066.3  856.29  5072.7  858.07  5103.1  860.21
  5108.3  858.37  5124.1  860.30  5197.3  861.57  5262.6  866.97  5323.2  872.80
  5360.0  886.17  5365.2  883.54  5370.9  885.90  5407.1  889.45  5476.8  890.62
#Mann=5,-1,0
  4435.5    0.05       0  4792.5    0.12       0  4991.4    0.07       0
  5004.1    0.12       0  5262.6    0.05       0
Bank Sta=4991.4,5004.1
Exp/Cntr=0.3,0.1

Type RM Length L Ch R = 1,97794,477,477,477
BEGIN DESCRIPTION:
Oliver Creek 120.0
END DESCRIPTION:
XS GIS Cut Line= 3
      2270449.42      7110746.18      2270642.20      7110146.50
      2270665.55      7109688.91
#Sta/Elev= 30
  4540.9  871.14  4586.4  867.28  4694.5  861.33  4778.5  858.79  4813.5  855.73
  4853.6  852.52  4885.7  854.84  4967.6  856.75  4982.0  851.97  4999.1  841.33
  5007.6  841.12  5009.4  840.62  5020.5  841.12  5030.6  846.93  5040.9  849.76
  5046.2  848.88  5072.6  852.05  5115.6  853.01  5156.6  859.68  5209.2  859.27
  5217.4  858.39  5237.4  851.76  5247.4  851.90  5257.4  855.32  5287.5  857.50
  5317.5  852.48  5347.5  855.38  5367.6  852.76  5407.6  860.63  5629.0  863.09
#Mann=4,-1,0
  4540.9    0.05       0  4813.5    0.12       0  5007.6    0.07       0
  5020.5    0.12       0
Bank Sta=5007.6,5020.5
Exp/Cntr=0.3,0.1

Type RM Length L Ch R = 1,97317,940,940,940
BEGIN DESCRIPTION:
Oliver Creek 119.0
END DESCRIPTION:
XS GIS Cut Line= 4
      2270947.38      7110731.21      2270942.34      7110493.06
      2270873.32      7110089.84      2270657.72      7109443.96
#Sta/Elev= 30
  4778.5  879.32  4859.7  873.81  4869.7  871.42  4899.7  858.66  4936.5  855.14
  4949.7  852.16  4959.8  848.63  4969.8  842.88  4973.3  839.07  4975.1  838.57
  4986.3  839.07  5009.8  843.15  5015.7  848.13  5060.4  853.19  5120.8  853.09
  5222.7  857.41  5344.5  859.28  5510.0  858.85  5516.8  856.12  5522.1  856.99
  5573.2  850.46  5604.8  855.71  5611.6  858.33  5625.9  858.94  5921.1  862.49
  6025.0  865.40  6047.6  867.00  6079.3  873.15  6091.0  880.14  6106.7  883.73
#Mann=4,-1,0
  4778.5    0.05       0  4973.3    0.07       0  4986.3    0.05       0
  6025.0    0.05       0
Bank Sta=4973.3,4986.3
Exp/Cntr=0.3,0.1

Type RM Length L Ch R = 1,96377,592,592,592
BEGIN DESCRIPTION:
Oliver Creek 118.0
END DESCRIPTION:
XS GIS Cut Line= 3
      2271451.92      7110887.41      2271334.35      7109843.12
      2271345.21      7109614.16
#Sta/Elev= 30
  3925.3  866.94  3985.5  864.85  4033.4  863.12  4144.1  861.42  4697.6  855.18
  4737.8  852.73  4778.1  848.83  4828.4  848.31  4848.5  849.29  4868.6  847.13
  4898.8  849.39  4918.9  848.00  4949.1  847.71  4959.2  846.09  4969.3  842.57
  4975.2  839.24  4989.3  838.39  4992.7  836.81  4994.6  836.31  5006.0  836.81
  5009.3  839.18  5019.4  850.72  5029.4  858.52  5039.4  858.72  5059.4  866.54
  5074.7  869.30  5099.4  872.25  5139.5  880.01  5159.5  881.95  5205.4  882.47
#Mann=5,-1,0
  3925.3    0.05       0  3985.5    0.12       0  4992.7    0.07       0
  5006.0    0.12       0  5074.7    0.05       0
Bank Sta=4992.7,5006
Exp/Cntr=0.3,0.1

Type RM Length L Ch R = 1,95785,334,334,334
BEGIN DESCRIPTION:
Oliver Creek 117.0
END DESCRIPTION:
XS GIS Cut Line= 3
      2272020.76      7110287.87      2271675.71      7109803.50
      2271378.83      7109489.69
#Sta/Elev= 30
  4448.0  862.28  4583.4  860.55  4676.5  856.41  4813.7  852.85  4826.9  851.72
  4841.6  847.63  4877.3  845.26  4992.9  846.79  5007.6  843.74  5013.7  839.00
  5022.4  836.40  5043.2  835.65  5045.1  835.15  5056.5  835.65  5057.1  837.49
  5064.0  840.60  5078.1  844.50  5106.4  846.59  5148.9  855.03  5205.5  857.39
  5249.7  857.09  5290.5  858.75  5333.0  863.25  5354.0  868.13  5375.4  868.85
  5410.6  873.55  5424.8  874.44  5460.4  872.40  5467.3  874.00  5474.7  872.70
#Mann=5,-1,0
  4448.0    0.05       0  4676.5    0.12       0  5043.2    0.07       0
  5056.5    0.12       0  5249.7    0.05       0
Bank Sta=5043.2,5056.5
Exp/Cntr=0.3,0.1

Type RM Length L Ch R = 1,95451,512,512,512
BEGIN DESCRIPTION:
Oliver Creek 116.0
END DESCRIPTION:
XS GIS Cut Line= 4
      2272046.53      7110363.13      2271969.63      7109849.96
      2272004.59      7109538.00      2272420.42      7109304.72
#Sta/Elev= 30
  4481.1  864.19  4544.9  863.08  4803.3  854.03  4959.5  846.47  4967.5  839.48
  4972.6  839.30  4979.7  834.34  4982.3  834.30  4984.3  833.80  4997.5  834.30
  5000.0  835.70  5020.1  837.81  5037.2  841.53  5042.2  840.76  5060.3  844.73
  5080.5  844.61  5110.6  848.74  5127.4  852.18  5205.1  853.88  5271.6  855.29
  5403.4  854.63  5441.0  853.37  5462.7  851.57  5506.1  852.93  5543.7  852.28
  5668.1  856.13  5743.2  862.35  5765.1  866.40  5777.6  871.68  5790.7  873.72
#Mann=5,-1,0
  4481.1    0.05       0  4803.3    0.12       0  4982.3    0.07       0
  4997.5    0.12       0  5205.1    0.05       0
Bank Sta=4982.3,4997.5
Exp/Cntr=0.3,0.1

Type RM Length L Ch R = 1,94939,594,594,594
BEGIN DESCRIPTION:
Oliver Creek 115.0
END DESCRIPTION:
XS GIS Cut Line= 3
      2272252.53      7110233.20      2272359.17      7109739.59
      2272423.11      7109329.54
#Sta/Elev= 30
  4495.0  861.86  4621.0  857.34  4640.2  855.49  4738.1  853.17  4754.0  853.07
  4788.0  850.17  4795.0  848.80  4825.7  847.06  4866.6  840.77  4876.3  842.70
  4881.4  840.65  4897.3  841.53  4917.7  840.01  4958.7  840.75  4981.7  833.97
  4983.7  833.47  4996.9  833.97  5002.3  834.05  5028.1  847.26  5033.2  847.33
  5040.1  849.37  5096.0  852.50  5101.1  851.53  5220.1  855.76  5236.8  856.46
  5283.0  858.28  5311.8  860.82  5352.3  862.22  5384.2  865.68  5415.0  870.76
#Mann=7,-1,0
  4495.0    0.05       0  4738.1    0.12       0  4981.7    0.07       0
  4996.9    0.12       0  5220.1    0.05       0  5236.8    0.12       0
  5311.8    0.05       0
Bank Sta=4981.7,4996.9
Exp/Cntr=0.3,0.1

Type RM Length L Ch R = 1,94345,458,458,458
BEGIN DESCRIPTION:
Oliver Creek 114.0
END DESCRIPTION:
XS GIS Cut Line= 3
      2272927.01      7110280.02      2272894.18      7109709.56
      2272856.89      7109343.16
#Sta/Elev= 30
  4428.6  868.01  4653.7  856.63  4669.0  856.45  4709.1  851.78  4729.1  851.29
  4759.2  847.51  4799.2  845.93  4819.3  844.08  4826.7  842.30  4899.4  841.68
  4949.5  839.80  4959.5  840.31  4969.5  839.38  4981.8  832.97  4983.8  832.47
  4995.2  832.47  4997.2  832.97  5009.6  834.14  5019.7  837.22  5029.7  843.13
  5039.8  846.52  5059.9  848.68  5102.8  850.55  5140.3  853.64  5160.4  853.96
  5180.5  856.36  5190.5  856.56  5202.5  857.79  5325.8  860.67  5368.3  861.43
#Mann=5,-1,0
  4428.6    0.05       0  4653.7    0.12       0  4981.8    0.07       0
  4997.2    0.12       0  5325.8    0.05       0
Bank Sta=4981.8,4997.2
Exp/Cntr=0.3,0.1

Type RM Length L Ch R = 1,93887,946,946,946
BEGIN DESCRIPTION:
Oliver Creek 113.0
END DESCRIPTION:
XS GIS Cut Line= 4
      2273528.56      7109921.98      2273229.00      7109710.00
      2273031.18      7109636.83      2272850.98      7109316.31
#Sta/Elev= 30
  4633.7  875.76  4693.0  874.02  4699.1  871.11  4713.9  868.41  4720.0  865.21
  4734.8  860.68  4760.9  857.50  4835.8  850.41  4957.6  844.36  4963.9  842.98
  4978.5  835.90  4979.4  832.06  4981.4  831.56  4994.9  832.06  5015.9  834.54
  5022.0  837.33  5041.0  840.75  5046.3  839.97  5132.2  841.29  5157.2  840.76
  5171.3  839.13  5181.9  839.69  5193.0  842.99  5210.1  845.72  5241.6  845.66
  5253.8  847.36  5344.3  851.73  5393.4  855.76  5493.7  859.63  5579.3  861.90
#Mann=5,-1,0
  4633.7    0.05       0  4760.9    0.12       0  4979.4    0.07       0
  4994.9    0.12       0  5493.7    0.05       0
Bank Sta=4979.4,4994.9
Exp/Cntr=0.3,0.1

Type RM Length L Ch R = 1,92941,431,431,431
BEGIN DESCRIPTION:
Oliver Creek 111.0
END DESCRIPTION:
XS GIS Cut Line= 3
      2273811.30      7109613.86      2273633.92      7109446.78
      2272894.60      7109099.96
#Sta/Elev= 30
  4719.4  870.90  4759.2  869.41  4773.4  866.83  4830.0  861.90  4854.4  860.74
  4886.6  859.20  4893.5  857.75  4900.8  854.58  4907.7  852.88  4921.8  840.10
  4928.7  837.59  4935.1  830.60  4937.1  830.10  4950.7  830.60  4957.0  830.61
  4963.0  832.16  4970.7  831.00  4987.9  836.06  4993.5  834.88  5001.6  838.64
  5016.3  839.33  5045.8  838.09  5061.9  839.31  5067.9  841.24  5084.7  843.00
  5256.7  847.66  5432.4  852.84  5489.2  854.19  5512.1  853.99  5779.7  861.10
#Mann=5,-1,0
  4719.4    0.05       0  4854.4    0.12       0  4935.1    0.07       0
  4950.7    0.12       0  5256.7    0.05       0
Bank Sta=4935.1,4950.7
Exp/Cntr=0.3,0.1

Type RM Length L Ch R = 1,92510,448,448,448
BEGIN DESCRIPTION:
Oliver Creek 110.0
END DESCRIPTION:
XS GIS Cut Line= 3
      2274074.82      7109392.03      2273692.57      7109046.76
      2273096.09      7108608.62
#Sta/Elev= 30
  4484.9  866.35  4667.8  860.35  4688.7  858.22  4745.5  857.01  4765.7  854.12
  4809.0  852.87  4872.6  846.36  4880.0  843.37  4886.8  844.33  4894.2  841.89
  4901.0  842.89  4908.4  841.46  4915.2  841.84  4936.8  836.55  4957.8  835.95
  4978.4  830.24  4980.4  829.74  4994.0  830.24  5006.8  832.82  5015.2  838.27
  5025.9  838.77  5057.0  838.73  5100.9  842.31  5107.1  841.44  5157.3  841.87
  5265.0  846.36  5357.9  847.20  5514.5  852.20  5629.5  857.19  5740.1  866.33
#Mann=5,-1,0
  4484.9    0.05       0  4765.7    0.12       0  4978.4    0.07       0
  4994.0    0.12       0  5025.9    0.05       0
Bank Sta=4978.4,4994
Exp/Cntr=0.3,0.1

Type RM Length L Ch R = 1,92062,620,620,620
BEGIN DESCRIPTION:
Oliver Creek 109.0
END DESCRIPTION:
XS GIS Cut Line= 3
      2274320.05      7109220.59      2273951.28      7108729.51
      2273379.00      7108310.00
#Sta/Elev= 30
  4359.7  862.68  4453.6  861.10  4682.8  852.45  4703.6  850.20  4760.6  847.87
  4794.8  844.99  4839.0  842.69  4868.1  838.84  4874.4  839.25  4882.7  837.00
  4924.4  836.55  4953.5  833.23  4960.3  830.13  4962.3  829.63  4976.0  830.13
  4989.1  831.09  4996.8  833.15  5003.0  836.61  5017.7  836.81  5038.6  840.74
  5064.8  842.76  5261.8  845.80  5297.8  845.20  5410.6  848.66  5554.9  851.13
  5590.4  854.51  5619.7  862.22  5633.8  868.39  5646.8  871.05  5683.4  872.36
#Mann=5,-1,0
  4359.7    0.05       0  4794.8    0.12       0  4960.3    0.07       0
  4976.0    0.12       0  5064.8    0.05       0
Bank Sta=4960.3,4976
Exp/Cntr=0.3,0.1

Type RM Length L Ch R = 1,91442,311,311,311
BEGIN DESCRIPTION:
Oliver Creek 108.0
END DESCRIPTION:
XS GIS Cut Line= 3
      2274747.58      7109055.67      2274354.04      7108360.08
      2274147.36      7108024.17
#Sta/Elev= 30
  4200.8  864.59  4285.7  861.85  4469.0  851.48  4582.9  846.74  4711.4  843.04
  4885.2  840.54  4908.2  838.51  4931.2  834.51  4965.6  835.25  4988.6  830.22
  4995.1  830.19  4997.1  829.69  5011.0  830.19  5024.3  838.04  5055.1  835.42
  5070.5  837.79  5076.4  839.65  5082.3  844.82  5091.8  850.18  5097.7  850.69
  5113.1  857.00  5119.0  856.53  5128.5  859.42  5134.4  859.47  5149.8  865.89
  5177.0  868.25  5207.8  867.49  5258.4  869.74  5275.4  869.01  5394.4  871.00
#Mann=5,-1,0
  4200.8    0.05       0  4582.9    0.12       0  4995.1    0.07       0
  5011.0    0.12       0  5275.4    0.05       0
Bank Sta=4995.1,5011
Exp/Cntr=0.3,0.1

Type RM Length L Ch R = 1,91131,442,442,442
BEGIN DESCRIPTION:
Oliver Creek 107.0
END DESCRIPTION:
XS GIS Cut Line= 3
      2274851.75      7108923.30      2274607.41      7108209.78
      2274371.63      7107922.56
#Sta/Elev= 30
  4245.8  863.26  4259.9  862.87  4312.7  857.74  4449.9  849.06  4563.2  843.74
  4642.9  841.18  4746.1  839.60  4851.3  835.81  4904.6  835.15  4936.3  836.10
  4957.5  835.22  4968.1  832.81  4968.5  831.26  4970.5  830.76  4984.4  831.26
  5026.6  834.79  5034.5  838.03  5040.9  838.64  5048.8  845.61  5063.2  849.92
  5069.6  850.60  5077.3  855.51  5084.0  857.30  5147.9  867.04  5184.3  866.67
  5240.4  868.47  5261.2  867.44  5310.8  868.67  5325.1  867.72  5371.6  868.04
#Mann=5,-1,0
  4245.8    0.05       0  4563.2    0.12       0  4968.5    0.07       0
  4984.4    0.12       0  5184.3    0.05       0
Bank Sta=4968.5,4984.4
Exp/Cntr=0.3,0.1

Type RM Length L Ch R = 1,90689,413,413,413
BEGIN DESCRIPTION:
Oliver Creek 106.0
END DESCRIPTION:
XS GIS Cut Line= 3
      2274932.04      7108942.85      2275002.80      7108333.14
      2275300.98      7107955.72
#Sta/Elev= 30
  4386.2  864.15  4429.3  863.34  4459.5  861.58  4530.0  854.83  4576.0  851.48
  4620.6  849.73  4681.0  843.52  4741.4  840.85  4771.6  838.43  4801.8  838.07
  4833.0  835.56  4862.2  832.70  4912.6  831.23  4917.4  830.24  4919.4  829.74
  4934.0  830.24  5014.2  830.26  5020.6  833.17  5035.0  835.87  5063.9  836.47
  5099.2  835.65  5113.6  836.91  5163.3  837.80  5177.7  839.97  5199.2  840.58
  5341.2  850.21  5355.6  852.55  5370.1  853.39  5411.8  860.05  5481.0  864.40
#Mann=5,-1,0
  4386.2    0.05       0  4833.0    0.12       0  4917.4    0.07       0
  4934.0    0.12       0  5199.2    0.05       0
Bank Sta=4917.4,4934
Exp/Cntr=0.3,0.1

Type RM Length L Ch R = 1,90276,463,463,463
BEGIN DESCRIPTION:
Oliver Creek 105.0
END DESCRIPTION:
XS GIS Cut Line= 3
      2275066.60      7109027.45      2275298.89      7108580.28
      2275510.73      7107974.02
#Sta/Elev= 30
  4496.1  861.22  4571.8  859.02  4770.9  849.47  4808.7  846.82  4815.1  845.31
  4831.3  845.16  4842.9  842.11  4875.8  838.88  4897.9  838.13  4903.6  840.84
  4910.2  838.39  4925.7  836.81  4947.8  832.49  4989.0  830.31  4991.0  829.81
  5005.6  830.31  5041.6  830.65  5046.9  831.38  5053.3  834.27  5063.8  835.43
  5112.2  835.06  5134.7  836.60  5222.6  838.87  5290.0  839.43  5307.5  841.40
  5368.8  844.94  5424.0  849.52  5465.7  856.85  5496.7  860.16  5642.2  865.90
#Mann=5,-1,0
  4496.1    0.05       0  4989.0   0.033       0  5005.6    0.05       0
  5112.2    0.12       0  5368.8    0.05       0
Bank Sta=4989,5005.6
Exp/Cntr=0.3,0.1

Type RM Length L Ch R = 1,89813,510,510,510
BEGIN DESCRIPTION:
Oliver Creek 104.0
END DESCRIPTION:
XS GIS Cut Line= 4
      2275268.05      7109633.72      2275726.32      7108801.99
      2275680.33      7108379.31      2275598.28      7107879.49
#Sta/Elev= 30
  3696.7  864.88  3876.4  862.74  4430.1  850.80  4670.6  843.14  4757.1  838.70
  4769.0  836.93  4799.2  834.90  4839.4  833.67  4899.8  834.26  4945.1  833.00
  4960.1  831.11  4970.2  832.55  5082.8  830.34  5084.8  829.84  5099.4  830.34
  5101.2  831.88  5108.4  833.40  5117.1  837.31  5131.6  840.90  5151.9  841.99
  5169.7  845.09  5192.4  846.77  5231.4  851.88  5236.0  851.44  5253.2  855.26
  5273.5  858.14  5303.9  860.26  5395.1  862.62  5537.0  863.99  5578.0  867.53
#Mann=5,-1,0
  3696.7    0.05       0  5082.8   0.033       0  5099.4    0.05       0
  5117.1    0.12       0  5231.4    0.05       0
Bank Sta=5082.8,5099.4
Exp/Cntr=0.3,0.1

Type RM Length L Ch R = 1,89303,443,443,443
BEGIN DESCRIPTION:
Oliver Creek 103.0
END DESCRIPTION:
XS GIS Cut Line= 3
      2275363.06      7109599.93      2276129.00      7108460.00
      2276150.58      7107997.76
#Sta/Elev= 30
  3626.2  862.96  3674.3  863.76  3681.0  862.65  3831.0  860.98  3855.0  859.29
  3891.0  859.74  4329.0  848.50  4575.0  844.72  4688.6  839.72  4761.1  837.19
  4770.0  835.30  4776.0  835.86  4797.1  832.89  4838.5  832.40  5031.2  830.49
  5033.2  829.99  5047.9  830.49  5049.6  832.19  5059.6  834.03  5069.6  838.73
  5099.7  846.13  5105.7  849.60  5119.7  854.38  5139.7  859.32  5149.7  860.28
  5219.8  861.76  5229.8  860.72  5323.1  860.35  5430.0  862.41  5462.3  861.87
#Mann=5,-1,0
  3626.2    0.05       0  4688.6    0.12       0  4838.5    0.05       0
  5031.2   0.033       0  5047.9    0.05       0
Bank Sta=5031.2,5047.9
Exp/Cntr=0.3,0.1

Type RM Length L Ch R = 1,88860,557,557,557
BEGIN DESCRIPTION:
Oliver Creek 102.0
END DESCRIPTION:
XS GIS Cut Line= 5
      2275510.43      7109531.88      2275677.75      7109276.78
      2276472.94      7108712.56      2276558.56      7108505.55
      2276364.34      7107849.10
#Sta/Elev= 30
  3719.9  861.00  3901.5  857.97  4353.9  842.77  4460.9  841.43  4467.9  840.52
  4511.4  839.45  4582.7  838.97  4627.0  836.81  4668.8  837.01  4683.6  835.93
  4704.5  836.44  4713.2  835.59  4743.8  835.50  4867.5  831.58  4897.9  830.07
  4899.9  829.57  4914.6  830.07  5089.3  830.32  5111.9  833.66  5121.8  835.99
  5143.5  844.85  5154.3  848.04  5159.7  852.00  5165.1  854.01  5183.6  858.91
  5189.0  859.28  5314.5  858.23  5438.4  855.74  5552.6  855.85  5908.6  861.82
#Mann=5,-1,0
  3719.9    0.05       0  4743.8    0.12       0  4867.5    0.05       0
  4897.9   0.033       0  4914.6    0.05       0
Bank Sta=4897.9,4914.6
Exp/Cntr=0.3,0.1

Type RM Length L Ch R = 1,88303,598,598,598
BEGIN DESCRIPTION:
Oliver Creek 101.0
END DESCRIPTION:
XS GIS Cut Line= 4
      2277575.84      7109903.93      2277543.15      7109617.12
      2276958.84      7108629.61      2276407.62      7107823.92
#Sta/Elev= 30
  3563.9  879.16  3618.2  878.51  3708.8  874.44  3728.9  872.72  3760.4  866.90
  3809.4  863.57  3844.8  863.75  4000.3  856.51  4102.6  854.61  4118.1  852.30
  4145.5  846.02  4161.1  845.97  4204.0  840.09  4321.0  833.03  4386.0  832.29
  4443.8  830.30  4986.0  831.22  5075.9  830.18  5077.9  829.68  5094.0  830.18
  5099.8  830.55  5114.7  836.97  5120.8  835.44  5157.0  840.36  5258.3  844.75
  5365.9  848.60  5467.5  847.11  5575.2  847.86  5790.5  857.29  5976.2  861.78
#Mann=5,-1,0
  3563.9    0.05       0  4118.1    0.12       0  4386.0    0.05       0
  5075.9   0.033       0  5094.0    0.05       0
Bank Sta=5075.9,5094
Exp/Cntr=0.3,0.1

Type RM Length L Ch R = 1,87705,1614,1614,1614
BEGIN DESCRIPTION:
Oliver Creek 100.0
END DESCRIPTION:
XS GIS Cut Line= 3
      2277722.86      7109673.55      2277429.00      7108860.00
      2276593.44      7107680.46
#Sta/Elev= 30
  4131.4  871.30  4154.3  869.38  4159.6  870.87  4190.3  867.57  4394.3  861.00
  4542.3  857.52  4698.7  856.02  4730.6  856.55  4815.6  854.55  4826.3  853.68
  4838.4  849.68  4858.2  845.16  4869.0  840.97  4889.1  840.60  4900.7  835.98
  4919.7  830.30  5369.3  831.12  5568.2  830.14  5570.2  829.64  5586.3  830.14
  5692.9  832.48  5793.0  836.83  5878.7  837.76  5915.5  841.05  5972.2  841.94
  6108.8  849.18  6180.2  855.08  6236.8  857.76  6245.4  859.60  6441.9  861.97
#Mann=3,-1,0
  4131.4    0.05       0  5568.2   0.033       0  5586.3    0.05       0
Bank Sta=5568.2,5586.3
Exp/Cntr=0.3,0.1

Type RM Length L Ch R = 1,86091,127,127,127
BEGIN DESCRIPTION:
Oliver Creek 99.0
END DESCRIPTION:
XS GIS Cut Line= 5
      2277818.72      7109529.52      2278045.74      7108907.04
      2277994.22      7107759.48      2277996.42      7107685.47
      2276855.15      7107204.55
#Sta/Elev= 30
  3188.7  865.15  3560.7  855.67  4058.5  849.45  4088.6  847.14  4108.3  847.35
  4128.6  845.50  4318.8  838.16  4579.1  830.34  5092.9  831.42  5375.1  830.39
  5440.7  832.08  5459.0  831.63  5459.1  829.91  5461.1  829.41  5477.4  829.91
  5535.6  831.24  5559.3  836.12  5564.8  833.42  5581.3  836.15  5588.5  835.88
  5593.9  833.37  5612.2  837.11  5635.5  836.28  5646.8  839.16  5665.1  841.26
  5678.9  846.41  5741.7  850.74  6015.3  857.27  6037.0  859.32  6312.5  861.89
#Mann=3,-1,0
  3188.7    0.05       0  5459.1   0.033       0  5477.4    0.05       0
Bank Sta=5459.1,5477.4
Exp/Cntr=0.3,0.1

Type RM Length L Ch R = 1,85964,182,182,182
BEGIN DESCRIPTION:
Oliver Creek 98.8
END DESCRIPTION:
XS GIS Cut Line= 6
      2277879.89      7109663.27      2278171.79      7108896.08
      2278121.88      7107760.02      2278117.71      7107338.18
      2277845.72      7107107.16      2277848.33      7106213.48
#Sta/Elev= 30
  3042.0  866.57  3252.3  861.38  3562.1  862.95  3586.8  860.68  3592.2  863.06
  3616.9  863.00  3671.8  860.04  3677.2  862.95  3701.9  863.06  3726.7  860.51
  3732.0  862.92  3751.4  860.59  3756.8  862.95  3781.6  860.66  3786.9  862.67
  3811.7  860.79  3817.0  862.73  4179.2  863.64  5390.0  861.20  5617.8  862.76
  5695.8  861.53  5795.9  854.30  5937.3  853.75  5939.3  853.25  5955.6  853.75
  6025.9  854.73  6055.9  861.55  6145.9  862.09  6225.9  866.82  6672.4  872.44
#Mann=3,-1,0
  3042.0    0.05       0  5937.3   0.033       0  5955.6    0.05       0
Bank Sta=5937.3,5955.6
Exp/Cntr=0.3,0.1

Type RM Length L Ch R = 1,85782,247,247,247
BEGIN DESCRIPTION:
Oliver Creek 98.5
END DESCRIPTION:
XS GIS Cut Line= 4
      2277980.82      7109735.92      2278354.77      7108909.33
      2278303.24      7107761.77      2278330.40      7107023.32
#Sta/Elev= 30
  2942.3  864.53  3376.8  852.77  3878.9  848.91  4079.1  849.74  4179.2  847.88
  4249.3  844.80  4308.4  838.63  4528.0  828.81  4589.6  825.03  4756.6  823.21
  4789.8  825.19  4827.6  823.72  4909.9  821.62  4940.0  814.85  4960.0  804.40
  5012.7  801.45  5014.7  800.95  5031.1  801.45  5070.1  815.50  5100.1  821.93
  5139.9  825.48  5208.6  835.86  5250.2  845.26  5300.2  847.96  5320.2  846.16
  5564.2  848.59  5610.4  849.51  5640.5  854.48  5670.5  849.64  5737.2  848.46
#Mann=7,-1,0
  2942.3    0.05       0  4528.0    0.12       0  4827.6    0.05       0
  5012.7   0.033       0  5031.1    0.05       0  5139.9    0.12       0
  5208.6    0.05       0
Bank Sta=5012.7,5031.1
Exp/Cntr=0.3,0.1

Type RM Length L Ch R = 1,85535,317,317,317
BEGIN DESCRIPTION:
Mapping XS d8a5805e
END DESCRIPTION:
XS GIS Cut Line= 3
      2278933.31      7108582.39      2278597.08      7107960.11
      2278397.80      7107105.44
#Sta/Elev= 30
  4087.5  848.10  4270.9  846.86  4306.2  844.09  4342.2  837.90  4458.4  829.68
  4495.2  828.11  4599.9  825.77  4937.0  821.97  4984.7  814.43  5000.3  804.21
  5001.4  802.03  5003.4  801.53  5019.8  802.03  5027.3  807.95  5032.4  806.58
  5041.4  812.98  5051.6  816.96  5061.9  818.15  5092.7  815.98  5226.2  821.23
  5324.2  830.35  5383.1  838.20  5425.7  839.32  5452.1  844.20  5558.5  846.95
  5585.6  851.46  5601.0  848.72  5606.2  850.63  5636.9  847.21  5672.4  847.32
#Mann=7,-1,0
  4087.5    0.05       0  4458.4    0.12       0  4495.2    0.05       0
  4599.9     0.1       0  5001.4    0.05       0  5019.8     0.1       0
  5324.2    0.05       0
Bank Sta=5001.4,5019.8
Exp/Cntr=0.3,0.1

Type RM Length L Ch R = 1,85218,518,518,518
BEGIN DESCRIPTION:
Oliver Creek 98.0
END DESCRIPTION:
XS GIS Cut Line= 3
      2279431.15      7108545.92      2278728.84      7107549.93
      2278226.28      7106618.80
#Sta/Elev= 30
  3781.3  847.46  3987.5  843.90  4433.4  828.18  4777.3  819.73  4877.6  821.86
  4900.1  812.56  4906.2  806.61  4914.3  805.79  4921.0  808.97  4927.1  803.65
  4935.8  805.35  4962.3  801.22  4964.3  800.72  4980.7  801.22  4992.4  806.11
  5007.9  801.89  5013.6  804.57  5051.7  804.64  5067.9  810.01  5117.4  810.74
  5177.3  823.10  5284.6  832.86  5434.3  845.50  5516.2  845.16  5554.3  839.98
  5590.8  844.06  5613.6  839.24  5625.7  844.91  5680.0  848.47  6058.1  851.87
#Mann=5,-1,0
  3781.3    0.05       0  4777.3     0.1       0  4962.3    0.05       0
  4980.7     0.1       0  5284.6    0.05       0
#XS Ineff=2,0
    0.00 4873.00  833.79               0
Permanent Ineff=
       F       F
Bank Sta=4962.3,4980.7
Exp/Cntr=0.3,0.1

Type RM Length L Ch R = 1,84700,621,621,621
BEGIN DESCRIPTION:
Oliver Creek 97.0
END DESCRIPTION:
XS GIS Cut Line= 3
      2279386.84      7108366.01      2279138.56      7107309.11
      2278668.32      7106513.57
#Sta/Elev= 30
  3915.2  843.50  4144.2  835.12  4229.1  833.81  4548.0  818.72  4722.5  815.89
  4800.9  811.74  4890.9  813.77  4933.3  811.73  4989.7  811.96  5003.3  809.78
  5007.7  803.76  5013.5  805.01  5029.2  802.12  5050.6  801.83  5057.1  799.73
  5059.1  799.23  5075.5  799.73  5087.7  811.42  5093.5  812.15  5109.1  818.57
  5183.3  824.25  5220.6  831.22  5226.2  834.09  5241.8  836.16  5247.6  839.05
  5306.1  844.80  5364.7  846.30  5497.3  845.67  5854.3  852.77  5925.0  852.17
#Mann=5,-1,0
  3915.2    0.05       0  4722.5     0.1       0  5057.1    0.05       0
  5075.5     0.1       0  5220.6    0.05       0
#XS Ineff=2,0
    0.00 4807.70  829.68               0
Permanent Ineff=
       F       F
Bank Sta=5057.1,5075.5
Exp/Cntr=0.3,0.1

Type RM Length L Ch R = 1,84079,584,584,584
BEGIN DESCRIPTION:
Mapping XS ec51a29d
END DESCRIPTION:
XS GIS Cut Line= 3
      2279806.42      7107697.49      2279472.75      7106605.38
      2279217.80      7106385.68
#Sta/Elev= 30
  4382.3  838.34  4496.6  835.79  4536.5  828.93  4598.9  823.81  4665.8  818.51
  4731.4  810.34  4829.3  809.82  4923.4  813.64  4938.6  808.25  4944.3  800.37
  4945.5  797.01  4947.5  796.51  4964.0  797.01  4965.2  798.70  4996.6  803.62
  5009.4  808.61  5017.5  809.13  5037.0  804.00  5059.3  804.54  5075.0  808.37
  5080.3  805.50  5090.7  806.30  5107.8  810.89  5132.5  808.90  5178.7  816.02
  5277.0  815.42  5580.7  820.26  5615.9  825.81  5679.5  842.43  5860.8  844.61
#Mann=4,-1,0
  4382.3    0.05       0  4598.9    0.12       0  4945.5    0.05       0
  4964.0    0.05       0
Bank Sta=4945.5,4964
Exp/Cntr=0.3,0.1

Type RM Length L Ch R = 1,83495,92,92,92
BEGIN DESCRIPTION:
Oliver Creek 95.0
END DESCRIPTION:
XS GIS Cut Line= 4
      2280356.72      7107368.71      2280185.28      7106988.94
      2280028.55      7106894.81      2279324.74      7106381.18
#Sta/Elev= 30
  4400.5  824.69  4555.6  822.65  4747.9  816.30  4952.8  809.36  4965.6  807.59
  4975.3  802.17  4981.1  801.64  4990.6  795.37  4992.6  794.87  5009.1  795.37
  5011.1  797.40  5017.3  797.21  5038.2  801.88  5051.8  808.32  5088.4  811.62
  5167.9  811.20  5274.5  816.38  5667.9  821.59  5697.0  823.13  5711.7  828.05
  5732.6  831.14  5741.1  834.51  5747.2  833.88  5761.9  839.62  5768.1  838.60
  5776.6  840.30  5782.8  838.66  5791.3  841.14  5812.1  842.46  5871.3  842.89
#Mann=5,-1,0
  4400.5    0.05       0  4747.9    0.12       0  4990.6    0.07       0
  5009.1    0.12       0  5051.8    0.05       0
Bank Sta=4990.6,5009.1
Exp/Cntr=0.3,0.1

Type RM Length L Ch R = 1,83403,624,624,624
BEGIN DESCRIPTION:
Oliver Creek 94.0
END DESCRIPTION:
XS GIS Cut Line= 4
      2280682.22      7107143.00      2280280.77      7106876.09
      2280053.86      7106813.23      2279280.51      7106196.32
#Sta/Elev= 30
  4299.7  818.78  4399.0  815.82  4426.1  817.22  4456.2  816.57  4483.7  813.74
  4549.3  815.20  4714.7  814.56  4861.1  811.18  4895.4  809.10  4900.6  810.23
  4918.5  807.78  4969.2  805.50  4974.4  803.32  5001.5  798.19  5007.9  794.42
  5009.9  793.92  5026.4  794.42  5030.1  800.38  5036.5  807.30  5044.6  811.65
  5091.1  813.69  5106.9  813.68  5251.1  817.09  5385.6  817.83  5613.0  821.81
  5741.1  825.68  5749.1  826.19  5755.5  828.42  5805.2  826.92  6006.5  840.92
#Mann=5,-1,0
  4299.7    0.05       0  5007.9   0.033       0  5026.4    0.05       0
  5091.1    0.12       0  5106.9    0.05       0
Bank Sta=5007.9,5026.4
Exp/Cntr=0.3,0.1

Type RM Length L Ch R = 1,82779,754,754,754
BEGIN DESCRIPTION:
Oliver Creek 93.0
END DESCRIPTION:
XS GIS Cut Line= 3
      2280877.57      7107156.07      2280558.83      7106459.54
      2280305.43      7105983.48
#Sta/Elev= 30
  4234.0  821.44  4306.7  817.63  4341.9  818.45  4372.6  815.01  4508.5  810.17
  4582.9  810.86  4691.6  807.08  4767.2  811.13  4834.5  807.67  4864.7  807.94
  4887.7  804.50  4944.8  806.99  4955.5  804.85  4962.3  797.96  4967.8  797.83
  4976.0  794.09  4978.0  793.59  4994.6  794.09  4997.0  796.20  5002.6  796.20
  5007.7  802.26  5013.4  802.45  5029.7  811.70  5304.0  816.33  5360.9  819.64
  5435.8  832.59  5441.4  836.75  5452.1  837.57  5457.7  835.90  5539.3  838.68
#Mann=5,-1,0
  4234.0    0.05       0  4582.9    0.12       0  4976.0    0.07       0
  4994.6    0.12       0  5360.9    0.05       0
Bank Sta=4976,4994.6
Exp/Cntr=0.3,0.1

Type RM Length L Ch R = 1,82025,453,453,453
BEGIN DESCRIPTION:
Oliver Creek 92.5
END DESCRIPTION:
XS GIS Cut Line= 3
      2281254.20      7107243.67      2281255.94      7106583.88
      2281297.15      7105854.44
#Sta/Elev= 30
  4340.2  826.29  4513.9  821.55  4533.9  822.45  4853.9  812.31  4913.9  812.68
  4933.9  809.26  4941.5  811.52  4953.9  811.83  4963.9  805.74  4973.9  797.08
  4983.9  793.92  4984.6  791.50  4986.6  791.00  5003.2  791.50  5004.4  793.08
  5013.9  794.20  5033.9  804.97  5054.0  806.55  5124.1  805.36  5154.1  802.22
  5194.2  800.99  5214.2  803.12  5244.3  801.31  5264.3  805.37  5294.3  826.93
  5311.1  831.36  5364.5  835.89  5493.6  834.59  5715.0  839.64  5730.6  838.38
#Mann=5,-1,0
  4340.2    0.05       0  4941.5    0.12       0  4984.6    0.07       0
  5003.2    0.12       0  5311.1    0.05       0
Bank Sta=4984.6,5003.2
Exp/Cntr=0.3,0.1

Type RM Length L Ch R = 1,81572,536,536,536
BEGIN DESCRIPTION:
Oliver Creek 92.0
END DESCRIPTION:
XS GIS Cut Line= 3
      2281470.35      7107217.66      2281561.50      7106359.99
      2281535.45      7105689.00
#Sta/Elev= 30
  4137.5  825.15  4195.5  824.11  4235.7  821.27  4296.1  821.44  4316.2  819.52
  4658.1  809.81  4818.3  807.87  4839.3  808.40  4926.8  804.19  4931.8  805.22
  4959.8  804.74  4969.8  803.34  4979.9  797.67  4980.5  789.97  4982.5  789.47
  4999.3  789.97  5000.0  792.52  5010.0  796.08  5020.0  802.14  5080.1  822.82
  5100.1  827.10  5126.9  828.90  5160.1  827.65  5189.2  822.93  5200.1  827.42
  5220.2  829.03  5290.2  829.23  5480.4  838.28  5510.4  837.40  5671.5  842.86
#Mann=5,-1,0
  4137.5    0.05       0  4818.3    0.12       0  4980.5    0.07       0
  4999.3    0.12       0  5126.9    0.05       0
Bank Sta=4980.5,4999.3
Exp/Cntr=0.3,0.1

Type RM Length L Ch R = 1,81036,1035,1035,1035
BEGIN DESCRIPTION:
Oliver Creek 91.0
END DESCRIPTION:
XS GIS Cut Line= 3
      2281729.01      7107259.97      2282081.30      7106415.83
      2282255.82      7105903.33
#Sta/Elev= 30
  4085.3  826.70  4099.9  824.68  4129.1  823.21  4323.7  814.89  4407.4  813.96
  4460.4  810.96  4613.6  808.56  4749.5  807.55  4778.8  804.25  4850.2  802.78
  4855.6  804.35  4865.5  804.60  4908.8  801.10  4927.1  804.04  4973.8  800.99
  4980.1  798.48  4985.6  789.99  4987.6  789.49  5004.4  789.99  5004.6  791.37
  5027.3  798.57  5036.0  802.83  5041.3  805.92  5048.4  815.59  5072.6  828.42
  5115.2  831.88  5130.1  831.87  5166.7  835.25  5380.9  836.37  5541.4  840.28
#Mann=5,-1,0
  4085.3    0.05       0  4613.6    0.12       0  4985.6    0.07       0
  5004.4    0.12       0  5115.2    0.05       0
Bank Sta=4985.6,5004.4
Exp/Cntr=0.3,0.1

Type RM Length L Ch R = 1,80001,511,511,511
BEGIN DESCRIPTION:
Oliver Creek 90.0
END DESCRIPTION:
XS GIS Cut Line= 3
      2283322.66      7107334.21      2283107.45      7107004.87
      2283029.00      7106209.96
#Sta/Elev= 30
  4159.7  824.12  4260.3  821.56  4287.7  818.61  4332.0  816.90  4367.8  812.45
  4511.2  806.17  4598.2  803.71  4759.0  802.19  4788.0  805.93  4793.0  804.13
  4809.2  805.11  4863.8  802.44  4919.8  800.66  4939.9  794.54  4948.2  785.65
  4950.6  785.15  4971.7  785.65  4990.1  789.24  4995.3  792.35  5000.3  789.99
  5010.2  796.19  5030.3  801.51  5060.4  803.22  5090.6  801.86  5096.5  805.89
  5130.8  818.41  5177.3  820.92  5202.6  822.68  5271.5  823.11  5351.9  827.05
#Mann=5,-1,0
  4159.7    0.05       0  4863.8    0.12       0  4948.2    0.07       0
  4971.7    0.12       0  5177.3    0.05       0
Bank Sta=4948.2,4971.7
Exp/Cntr=0.3,0.1

Type RM Length L Ch R = 1,79490,681,681,681
BEGIN DESCRIPTION:
Oliver Creek 89.0
END DESCRIPTION:
XS GIS Cut Line= 3
      2283797.16      7107063.54      2283536.60      7106458.46
      2283173.33      7105905.99
#Sta/Elev= 30
  4342.9  827.61  4556.1  817.68  4608.3  812.05  4738.7  803.78  4831.3  802.97
  4878.3  801.54  4907.3  798.66  4945.6  799.41  4954.4  796.42  4959.8  798.72
  4977.4  786.53  4979.7  786.03  5000.9  786.53  5006.1  789.52  5021.2  791.74
  5027.2  787.80  5035.8  791.21  5042.3  797.08  5048.3  793.52  5057.4  799.30
  5071.7  801.60  5198.1  802.47  5274.3  804.24  5280.3  807.12  5337.5  808.70
  5352.6  809.93  5358.9  813.56  5367.7  815.15  5382.8  816.03  5662.9  819.55
#Mann=5,-1,0
  4342.9    0.05       0  4608.3    0.12       0  4977.4    0.07       0
  5000.9    0.12       0  5198.1    0.05       0
Bank Sta=4977.4,5000.9
Exp/Cntr=0.3,0.1
