HEC-RAS study COTTONWOOD BR AT DENTON.prj: COTTONWOOD BR AT DENTON Base Level Engineering

--- COTTONWOOD BR AT DENTON.g01 (geometry) --- (continued)

Type RM Length L Ch R = 1 ,27790   ,209,209,209
BEGIN DESCRIPTION:
COTTONWOOD BR AT DENTON 46.4
END DESCRIPTION:
XS GIS Cut Line= 4
       2416248.2      7032909.96      2416557.39       7032612.9
      2416860.48      7032318.89      2417524.09      7031921.94
#Sta/Elev= 30
  4282.4   555.4  4311.2   553.1  4353.5  555.31  4466.7   553.2  4502.3  546.61
  4579.9  542.88  4834.6  541.07  4912.3  537.36  4961.9  528.88  4995.2  527.97
  4996.6  527.47  5004.8  527.97    5061  538.47  5139.3   542.9  5532.2  544.03
  5664.4     549  5670.3  551.84  5685.8  551.21  5707.2  554.72  5722.8   553.8
  5728.6  556.51  5744.2  555.61  5765.6   558.7  5781.1  557.85    5787  560.32
  5802.5  559.54  5808.4  561.87  5839.5  562.05  5845.3  564.13  5906.7  562.71
#Mann= 3 ,-1 , 0
  4282.4     .05       0  4995.2    .033       0  5004.8     .05       0
Bank Sta=4995.2,5004.8
XS Rating Curve= 0 ,0
Exp/Cntr=0.3,0.1

Type RM Length L Ch R = 1 ,27581   ,36,36,36
BEGIN DESCRIPTION:
COTTONWOOD BR AT DENTON 46.2
END DESCRIPTION:
XS GIS Cut Line= 4
      2416484.63      7033310.05      2416672.56      7032794.76
      2416948.38      7032488.63       2417263.6      7032176.44
#Sta/Elev= 30
  4174.9  550.52  4209.3  550.47  4405.2  544.21  4483.6   543.2  4504.9  538.79
  4515.6  537.81  4547.3  542.54  4752.7  546.27  4781.1  544.81    4802  540.29
  4816.2  542.12  4844.6  542.12  4851.4  540.75  4929.8  537.18  4985.9  528.13
  4995.2  527.85  4996.6  527.35  5004.8  527.85    5036  528.99  5050.2  530.99
  5071.1  536.58  5085.3  538.66  5149.1   543.1  5156.1  544.57  5163.2   544.1
  5170.3   545.7  5255.1  550.96  5410.7  558.56  5417.8  557.83  5579.1  559.24
#Mann= 4 ,-1 , 0
  4174.9    .075       0  4209.3     .05       0  4995.2    .033       0
  5004.8     .05       0
Bank Sta=4995.2,5004.8
XS Rating Curve= 0 ,0
Exp/Cntr=0.3,0.1

Type RM Length L Ch R = 1 ,27545   ,28,28,28
BEGIN DESCRIPTION:
COTTONWOOD BR AT DENTON 46.0
END DESCRIPTION:
XS GIS Cut Line= 4
      2416621.03      7033328.24       2416754.4      7032831.13
        2416939.      7032520.57      2417275.71      7032182.52
#Sta/Elev= 30
  4233.3  549.33  4282.1  549.08  4490.3  544.17  4542.1  537.34  4573.1  541.99
  4728.4  543.87  4766.8  539.89  4788.2  542.71  4819.1  543.05  4846.6  539.87
  4920.7  537.61  4970.3  529.39  4995.2  527.76  4996.6  527.26  5004.8  527.76
  5037.5  529.78  5086.7  539.16  5180.4  546.65  5187.5  549.21  5222.8  550.11
  5229.9  552.86    5237   551.5  5265.2  553.31  5272.3  555.83  5279.4  554.19
  5300.6  556.46  5314.7  554.25  5321.8  556.25  5364.2  557.84  5586.4  559.07
#Mann= 4 ,-1 , 0
  4233.3    .075       0  4282.1     .05       0  4995.2    .033       0
  5004.8     .05       0
Bank Sta=4995.2,5004.8
XS Rating Curve= 0 ,0
Exp/Cntr=0.3,0.1

Type RM Length L Ch R = 1 ,27517   ,161,161,161
BEGIN DESCRIPTION:
COTTONWOOD BR AT DENTON 45.8
END DESCRIPTION:
XS GIS Cut Line= 4
      2416663.48      7033322.12      2416824.11      7032803.85
      2416960.51      7032512.88      2417287.86      7032197.65
#Sta/Elev= 30
  4270.5  549.04  4312.3  548.56  4513.7  544.08  4534.4  540.86  4541.1  537.81
  4555.4  536.67  4597.3  541.58  4676.7  541.18  4714.5  538.17  4785.7  543.93
  4828.4  540.35  4916.7  538.34  4960.9  529.91  4995.2  527.61  4996.6  527.11
  5004.8  527.61  5046.1  531.25  5074.4  537.98  5120.1  543.76  5136.9  543.08
  5142.5  545.46  5177.8   547.4    5185   550.4  5220.2   551.2  5227.4     554
  5234.4  552.86  5241.6  554.93  5262.7  554.33  5269.9  557.03  5588.9  558.45
#Mann= 4 ,-1 , 0
  4270.5    .075       0  4312.3     .05       0  4995.2    .033       0
  5004.8     .05       0
Bank Sta=4995.2,5004.8
XS Rating Curve= 0 ,0
Exp/Cntr=0.3,0.1

Type RM Length L Ch R = 1 ,27356   ,531,531,531
BEGIN DESCRIPTION:
COTTONWOOD BR AT DENTON 45.0
END DESCRIPTION:
XS GIS Cut Line= 5
      2416911.99      7033013.03      2416990.82      7032809.91
      2417099.93      7032576.53      2417161.15      7032443.44
      2417444.37      7032165.38
#Sta/Elev= 30
  4679.9  545.46  4900.5  539.38  4909.8  535.25  4955.5   527.4  4995.2   526.4
  4996.5   525.9  5004.9   526.4  5008.1  530.39  5052.4  540.05  5092.5   542.8
  5184.1  542.52  5258.5   539.6    5264  537.42    5301  541.54  5437.2  538.74
  5444.2  541.06  5451.4  538.92  5479.6   539.4  5486.7  541.52  5522.1  540.62
  5529.1  543.01  5536.2  540.92  5543.2  542.97  5564.5  541.94  5571.5   544.5
  5606.9  543.68  5613.9  545.98  5656.4  543.26  5663.4  545.84  5698.8  546.54
#Mann= 3 ,-1 , 0
  4679.9     .05       0  4995.2    .033       0  5004.9     .05       0
Bank Sta=4995.2,5004.9
XS Rating Curve= 0 ,0
Exp/Cntr=0.3,0.1

Type RM Length L Ch R = 1 ,26825   ,422,422,422
BEGIN DESCRIPTION:
COTTONWOOD BR AT DENTON 44.0
END DESCRIPTION:
XS GIS Cut Line= 3
      2416909.15      7033358.44      2417582.02      7032969.43
      2418081.43      7032738.13
#Sta/Elev= 30
  4474.3  547.38  4543.7  545.05  4715.9   540.2  4774.4  537.21  4796.8  532.24
  4935.5  531.41  4970.8  525.69  4993.9  527.09  4995.1  523.58  4996.4  523.08
    5005  523.58  5021.7  524.16  5028.6   527.4  5086.3   536.2  5145.2  533.98
  5176.7  536.54  5182.5  533.97  5235.6  537.02  5241.3  533.69  5246.9  536.72
  5263.4  534.36  5391.5  538.08  5452.3  534.12  5480.7  535.75  5530.2  533.29
    5550  531.87  5600.9  527.63    5720  530.86  5761.2  538.92  5801.9  541.88
#Mann= 8 ,-1 , 0
  4474.3    .075       0  4543.7     .05       0  4796.8     .12       0
  4995.1     .07       0    5005     .12       0  5530.2     .05       0
    5550     .03       0    5720      .1       0
Bank Sta=4995.1,5005
XS Rating Curve= 0 ,0
Exp/Cntr=0.3,0.1

Type RM Length L Ch R = 1 ,26403   ,283,283,283
BEGIN DESCRIPTION:
COTTONWOOD BR AT DENTON 43.0
END DESCRIPTION:
XS GIS Cut Line= 3
      2416898.64      7033453.06      2417497.91      7033437.29
        2418544.        7033411.
#Sta/Elev= 30
  4319.3  548.49  4485.9   545.7  4709.8  537.66  4789.8  528.97  4889.9  527.43
  4959.9  527.88  4969.9  528.94  4989.9  526.93    4995   521.7  4996.4   521.2
    5005   521.7  5012.4   521.7  5019.9   524.6  5029.9  526.22  5099.9  526.58
  5139.9  530.21    5250  532.45    5260  529.35    5270  528.05    5300  533.95
  5406.5  535.53  5490.1  537.98  5500.1  539.19  5520.1  536.78  5530.1  533.74
  5540.1  533.37  5560.1  538.44  5600.1  539.75  5850.2   540.8  5965.2  542.88
#Mann= 4 ,-1 , 0
  4319.3    .075       0  4485.9     .05       0    4995    .033       0
    5005     .05       0
Bank Sta=4995,5005
XS Rating Curve= 0 ,0
Exp/Cntr=0.3,0.1

Type RM Length L Ch R = 1 ,26120   ,270,270,270
BEGIN DESCRIPTION:
COTTONWOOD BR AT DENTON 42.8
END DESCRIPTION:
XS GIS Cut Line= 3
      2416909.14      7033663.33      2417865.88      7033652.81
       2418415.9      7033589.96
#Sta/Elev= 30
  4227.1  546.12    4277  545.66    4307  542.09  4404.8   540.7  4471.4  540.59
    4507  539.85    4527  537.89    4617  536.49    4637  532.51    4657  535.83
    4727  535.16    4737  533.78  4784.9  532.78    4907  531.85    4937  526.23
    4977  525.65  4988.5  521.09    4995  521.09  4996.4  520.59  5005.1  521.09
    5007  524.97    5017  526.13    5027  526.82    5067  524.43    5107  532.94
  5170.6  533.81  5358.1  534.68  5470.4  537.12  5670.2     539  5737.5  537.47
#Mann= 8 ,-1 , 0
  4227.1    .075       0  4404.8      .1       0  4471.4    .075       0
  4784.9     .05       0    4995     .05       0  5005.1     .05       0
  5170.6    .075       0  5470.4     .05       0
Bank Sta=4995,5005.1
XS Rating Curve= 0 ,0
Exp/Cntr=0.3,0.1

Type RM Length L Ch R = 1 ,25850   ,479,479,479
BEGIN DESCRIPTION:
COTTONWOOD BR AT DENTON 42.0
END DESCRIPTION:
XS GIS Cut Line= 3
      2417171.96      7034089.14      2417734.46       7033910.4
      2418295.45      7033627.28
#Sta/Elev= 30
  4360.1  540.72    4399  538.99  4493.4  539.85  4545.9  537.02  4574.8  537.46
  4614.6   537.7  4797.7  536.44  4837.6  535.13  4937.2  532.36  4950.1  529.22
  4955.7  529.22  4961.6  526.19  4977.8  524.33  4983.9  521.06    4995  521.06
  4996.4  520.56  5005.1  521.06  5006.2  524.89  5011.8  525.05  5034.1  523.54
  5112.1  523.53  5134.4  525.95    5140  528.84  5145.8  529.76  5156.7  530.25
  5162.3  534.11    5179  533.51  5189.2  535.23  5414.1  535.15  5578.7  538.09
#Mann= 8 ,-1 , 0
  4360.1    .075       0  4574.8     .05       0  4614.6    .075       0
  4837.6     .05       0    4995    .033       0  5005.1     .05       0
  5189.2    .075       0  5414.1     .05       0
Bank Sta=4995,5005.1
XS Rating Curve= 0 ,0
Exp/Cntr=0.3,0.1

Type RM Length L Ch R = 1 ,25371   ,765,765,765
BEGIN DESCRIPTION:
COTTONWOOD BR AT DENTON 41.0
END DESCRIPTION:
XS GIS Cut Line= 3
       2417450.6      7034304.65      2418013.07      7034057.59
      2418529.04        7034010.
#Sta/Elev= 30
  4268.8  540.07  4354.4  538.06  4474.6   538.8  4507.3  537.39  4572.9  536.59
  4590.2  535.65  4642.4  535.65  4660.2  536.56  4747.6  535.44  4758.5  535.96
    4788  534.06  4840.2  532.33    4875  527.84  4883.1  527.46  4919.2  523.21
  4949.3  522.05  4959.4  523.85  4969.4  523.59  4989.5  518.74  4994.8  518.74
  4996.3  518.24  5005.2  518.74  5009.6  522.32  5010.5  522.43  5079.9  528.75
  5209.9  533.05    5331  538.08  5381.2  545.02  5398.7  549.84  5401.3  549.84
#Mann= 6 ,-1 , 0
  4268.8    .075       0    4875     .05       0  4994.8    .033       0
  5005.2     .05       0  5010.5     .12       0  5209.9     .05       0
Bank Sta=4994.8,5005.2
XS Rating Curve= 0 ,0
Exp/Cntr=0.3,0.1

Type RM Length L Ch R = 1 ,24606   ,536,536,536
BEGIN DESCRIPTION:
COTTONWOOD BR AT DENTON 40.0
END DESCRIPTION:
XS GIS Cut Line= 3
        2417950.      7035014.29      2418076.15      7034567.49
      2418601.83      7034020.79
#Sta/Elev= 30
  4580.8  537.98  4616.4  536.52  4637.4  537.98  4666.2  535.62  4907.4  533.75
  4917.8  533.75  4924.8   537.3    4930  532.29  4933.8  531.97  4980.1  526.53
  4990.5  523.02  4994.8  515.63  4996.3  515.13  5005.2  515.63  5011.3  515.63
  5037.2  520.43  5130.1  521.38  5208.1  527.53  5236.1  525.34  5314.1  526.86
  5391.8  526.32  5420.1  528.35  5560.4  533.27  5653.4  535.38    5710  538.42
  5717.2   540.2  5752.5  543.01  5766.6  545.31  5773.8  547.79  5803.5  551.86
#Mann= 5 ,-1 , 0
  4580.8     .05       0  4933.8     .12       0  4994.8     .07       0
  5005.2     .12       0  5560.4     .05       0
Bank Sta=4994.8,5005.2
XS Rating Curve= 0 ,0
Exp/Cntr=0.3,0.1

Type RM Length L Ch R = 1 ,24070   ,453,453,453
BEGIN DESCRIPTION:
COTTONWOOD BR AT DENTON 39.0
END DESCRIPTION:
XS GIS Cut Line= 3
      2418186.55      7035098.42      2418507.21      7034672.63
      2418800.88      7034274.07
#Sta/Elev= 30
  4428.6  538.28  4507.7  537.63  4543.1  534.88  4601.4  527.46  4643.1  525.43
  4672.2  518.25  4691.1  517.57  4736.8  518.21  4751.3   519.4  4757.6  521.55
  4836.7  521.85  4878.4  519.32  4907.5   520.4  4936.6  518.64  4942.9   520.5
  4951.2  519.12  4957.5  521.23  4972.1  520.21  4978.3  521.69  4992.9  518.66
  4994.8  515.55  4996.2  515.05  5005.3  515.55  5051.5  521.39  5164.2  527.16
  5214.3  530.44  5237.4  533.56  5243.6  532.68  5336.8  536.27  5456.7     539
#Mann= 5 ,-1 , 0
  4428.6     .05       0  4691.1     .12       0  4994.8     .07       0
  5005.3     .12       0  5336.8     .05       0
Bank Sta=4994.8,5005.3
XS Rating Curve= 0 ,0
Exp/Cntr=0.3,0.1

Type RM Length L Ch R = 1 ,23617   ,526,526,526
BEGIN DESCRIPTION:
COTTONWOOD BR AT DENTON 38.0
END DESCRIPTION:
XS GIS Cut Line= 3
      2418407.35      7035119.43      2418796.33      7034756.74
      2419147.21      7034473.94
#Sta/Elev= 30
    4377  535.78  4392.1   537.2    4399  535.74  4455.6  536.72  4476.6  535.16
    4484  536.36  4519.8  531.97  4564.6  528.18    4569  528.65  4575.8   525.5
  4604.2  522.65  4658.4  521.54  4823.5  520.98  4979.1  517.56  4993.5  517.07
  4994.8  511.45  4996.2  510.95  5005.3  511.45    5015  511.45  5022.3  517.11
  5028.7  515.09  5036.7  517.33  5051.1  517.46  5086.3  523.84  5135.9   536.4
  5180.1   537.6  5257.4  538.77  5271.8  537.43  5313.4  540.59  5359.5  540.44
#Mann= 7 ,-1 , 0
    4377     .05       0  4519.8     .12       0  4564.6     .05       0
  4658.4     .12       0  4994.8     .07       0  5005.3     .12       0
  5180.1     .05       0
Bank Sta=4994.8,5005.3
XS Rating Curve= 0 ,0
Exp/Cntr=0.3,0.1

Type RM Length L Ch R = 1 ,23091   ,341,341,341
BEGIN DESCRIPTION:
COTTONWOOD BR AT DENTON 37.0
END DESCRIPTION:
XS GIS Cut Line= 3
      2418233.89      7035208.81      2418833.13      7035108.94
      2419432.42      7035093.17
#Sta/Elev= 30
  4347.2   536.9  4585.5  534.52  4626.1  535.26  4673.1  533.21  4697.1     534
  4727.5  531.25    4734  528.69  4752.1  525.73  4778.2  521.03  4794.8  519.68
    4910  519.06  4950.1  514.74  4990.6  516.61  4994.7  510.88  4996.2  510.38
  5005.3  510.88  5010.6  510.88  5020.6  515.08  5030.6  516.08  5090.6  517.24
  5140.6  528.29  5150.6  527.75  5190.7  520.41  5210.7  519.86  5237.7  522.35
  5280.7  530.87  5310.7  534.45  5440.4   538.5  5500.8  540.41  5554.2  539.66
#Mann= 6 ,-1 , 0
  4347.2     .05       0  4752.1     .12       0  4994.7     .07       0
  5005.3     .12       0  5237.7     .05       0  5440.4    .075       0
Bank Sta=4994.7,5005.3
XS Rating Curve= 0 ,0
Exp/Cntr=0.3,0.1

Type RM Length L Ch R = 1 ,22750   ,502,502,502
BEGIN DESCRIPTION:
COTTONWOOD BR AT DENTON 36.0
END DESCRIPTION:
XS GIS Cut Line= 3
       2418181.3      7035434.86      2418833.13      7035387.55
      2419411.36      7035319.21
#Sta/Elev= 30
  4400.8  536.54  4528.8   535.2  4649.2  529.76  4674.7  527.81  4679.7  529.08
  4722.4  526.34  4808.9  522.26  4829.6  522.52  4839.7  521.38  4939.9   518.6
  4953.2  517.46    4970  513.82    4980  510.33    4990  514.04  4994.7  510.33
  4996.2  509.83  5005.3  510.33  5020.1  515.02  5080.7  515.18  5110.6  514.12
  5158.6   517.1  5163.6  516.53  5231.4  521.45    5244   521.4  5320.8  523.87
  5362.3  525.01  5520.9  533.66  5563.7  536.11  5614.1  540.64  5636.6  540.71
#Mann= 7 ,-1 , 0
  4400.8     .05       0  4722.4     .12       0  4994.7     .07       0
  5005.3     .12       0    5244     .05       0  5320.8     .12       0
  5520.9     .05       0
Bank Sta=4994.7,5005.3
XS Rating Curve= 0 ,0
Exp/Cntr=0.3,0.1

Type RM Length L Ch R = 1 ,22248   ,430,430,430
BEGIN DESCRIPTION:
COTTONWOOD BR AT DENTON 35.0
END DESCRIPTION:
XS GIS Cut Line= 3
      2417913.19      7035918.48        2419029.        7035710.
       2419315.4       7035640.2
#Sta/Elev= 30
  3864.5  534.09  3972.1  532.76    4023  535.82    4058  535.82  4100.3  539.25
  4152.9  532.26  4216.3  527.28    4316  525.02    4380  521.22  4389.2  517.13
  4399.4  516.95  4633.4  516.83  4655.9  518.61  4704.9  521.92  4735.1  517.34
    4868  516.12  4887.7  513.77  4915.5  512.64  4973.3  513.31  4989.4  512.39
  4994.7  509.11  4996.2  508.61  5005.3  509.11    5023  509.11  5040.8  516.32
  5059.6  520.55  5082.8  523.67  5101.3  526.49  5164.2  532.18  5294.4  539.82
#Mann= 8 ,-1 , 0
  3864.5    .075       0    4058     .05       0    4380     .03       0
  4655.9     .12       0  4994.7     .07       0  5005.3     .12       0
  5082.8     .05       0  5164.2     .12       0
Bank Sta=4994.7,5005.3
XS Rating Curve= 0 ,0
Exp/Cntr=0.3,0.1

Type RM Length L Ch R = 1 ,21818   ,442,442,442
BEGIN DESCRIPTION:
COTTONWOOD BR AT DENTON 34.0
END DESCRIPTION:
XS GIS Cut Line= 3
      2418317.94      7036622.91        2419079.        7036060.
      2419394.31      7035725.36
#Sta/Elev= 30
  4049.6  533.56  4143.4     532  4222.2   531.4  4366.8   526.7  4396.1  523.26
    4410  518.51    4775  517.22    4847  522.42  4859.4  517.53  4878.6  516.19
  4946.5  514.87  4994.6  508.62  4996.1  508.12  5005.5  508.62  5038.5  510.83
  5045.8  508.72  5052.6  511.08  5059.9  510.53  5066.8  514.36  5074.1  511.81
    5081  514.71  5088.3  513.46  5165.9  518.47  5236.7  526.64  5271.9  534.91
  5362.3  531.63  5378.3  532.28  5399.4  539.67  5443.1  541.45    5456  542.61
#Mann= 10 ,-1 , 0
  4049.6      .1       0  4143.4    .075       0  4222.2     .05       0
    4410     .03       0    4775     .05       0  4878.6     .12       0
  4994.6     .07       0  5005.5     .12       0  5362.3     .05       0
  5443.1      .1       0
Bank Sta=4994.6,5005.5
XS Rating Curve= 0 ,0
Exp/Cntr=0.3,0.1

Type RM Length L Ch R = 1 ,21376   ,457,457,457
BEGIN DESCRIPTION:
COTTONWOOD BR AT DENTON 33.0
END DESCRIPTION:
XS GIS Cut Line= 3
      2419222.12       7036575.6      2419458.69      7036254.92
      2419574.33      7035792.35
#Sta/Elev= 30
  4555.6  531.03  4568.7  530.61  4772.7   526.1  4793.5  524.55  4799.7  522.56
  4808.2  522.07  4814.4  520.33  4825.6  519.71  4864.5  517.15  4908.4   518.1
  4927.2  517.53  4959.2  515.04  4975.3  510.47  4990.1  508.35  4994.6  502.91
  4996.1  502.41  5005.5  502.91  5010.7  504.46  5021.7  502.91  5031.3  504.26
  5041.6  507.67  5093.2   514.8    5099  517.16  5122.8  520.93  5134.4  523.09
    5223  527.44    5289   528.1  5305.2  531.59  5319.9  532.28  5430.9   533.1
#Mann= 8 ,-1 , 0
  4555.6    .075       0  4568.7     .05       0  4825.6     .12       0
  4927.2     .05       0  4994.6    .033       0  5005.5     .05       0
  5122.8    .075       0    5223      .1       0
Bank Sta=4994.6,5005.5
XS Rating Curve= 0 ,0
Exp/Cntr=0.3,0.1

Type RM Length L Ch R = 1 ,20919   ,366,366,366
BEGIN DESCRIPTION:
COTTONWOOD BR AT DENTON 32.0
END DESCRIPTION:
XS GIS Cut Line= 3
      2419807.89      7036832.01        2419879.        7036310.
      2419891.21      7035708.85
#Sta/Elev= 30
  4477.5  525.72  4540.1  520.93  4570.4  520.97  4596.2   521.9    4641  519.92
  4695.2  519.19  4923.6   516.9  4933.7  511.13  4953.9  505.51  4963.1  504.37
  4974.1  501.54  4984.1  500.46  4994.2  503.96  4994.5  500.46    4996  499.96
  5005.5  500.46  5006.8   503.4  5034.3  503.28  5044.3  504.58  5074.3   512.4
  5094.3  516.16  5104.4  520.62  5124.4   520.6  5166.7  522.22  5494.4   527.5
  5544.4  526.21  5574.4  530.03  5584.5  530.75  5604.8  530.75  5605.6  530.75
#Mann= 6 ,-1 , 0
  4477.5     .05       0  4695.2    .075       0  4994.5     .07       0
  5005.5    .075       0  5166.7      .1       0  5604.8    .075       0
Bank Sta=4994.5,5005.5
XS Rating Curve= 0 ,0
Exp/Cntr=0.3,0.1

Type RM Length L Ch R = 1 ,20553   ,241,241,241
BEGIN DESCRIPTION:
COTTONWOOD BR AT DENTON 31.2
END DESCRIPTION:
XS GIS Cut Line= 3
      2420204.48      7036951.99      2420234.48      7036228.78
      2420244.42      7035993.63
#Sta/Elev= 30
  4407.9  523.04  4419.9  521.82  4468.5  520.32    4480  520.81  4610.1  520.57
  4650.1  518.95  4844.6  515.78  4920.3  513.46  4930.3   513.7  4940.4  511.51
  4960.4  505.14  4970.4   503.4  4980.4  502.65  4990.4  502.89  4994.5  500.01
    4996  499.51  5005.5  500.01  5010.4  501.92  5020.4  500.01  5060.5  502.14
  5070.5  504.25  5080.5  507.61  5090.5  508.79  5117.8  515.76  5122.8  515.47
  5128.6  516.75  5153.3  517.88  5190.6  517.54  5240.6  518.67  5367.1  523.26
#Mann= 6 ,-1 , 0
  4407.9     .05       0  4468.5    .075       0  4844.6     .05       0
  4994.5     .05       0  5005.5     .05       0  5153.3      .1       0
Bank Sta=4994.5,5005.5
XS Rating Curve= 0 ,0
Exp/Cntr=0.3,0.1

Type RM Length L Ch R = 1 ,20312   ,309,309,309
BEGIN DESCRIPTION:
COTTONWOOD BR AT DENTON 31.0
END DESCRIPTION:
XS GIS Cut Line= 3
      2420421.11      7036802.02      2420441.11      7036242.11
      2420451.11      7036005.49
#Sta/Elev= 30
  4555.9  523.58  4634.9  521.27    4678  521.45    4758  519.94  4788.1  518.44
  4818.1  514.42  4858.1  514.18  4878.1  515.96  4902.4  514.99  4915.1  512.99
  4920.1   513.4  4928.2  510.56  4948.1  506.07  4968.2  501.83  4988.2  501.85
  4994.5  498.79    4996  498.29  5005.6  498.79  5018.2  498.79  5028.2  500.86
  5038.2  501.57  5058.2  501.26  5078.3  505.35  5108.3  513.88  5128.3  516.48
  5158.3  518.18    5184  517.28  5218.4  517.98  5278.4  520.82    5353  522.17
#Mann= 5 ,-1 , 0
  4555.9    .075       0  4902.4     .05       0  4948.1    .075       0
  4994.5     .07       0  5005.6    .075       0
Bank Sta=4994.5,5005.6
XS Rating Curve= 0 ,0
Exp/Cntr=0.3,0.1

Type RM Length L Ch R = 1 ,20003   ,456,456,456
BEGIN DESCRIPTION:
COTTONWOOD BR AT DENTON 30.0
END DESCRIPTION:
XS GIS Cut Line= 3
      2420664.41      7037101.92        2420729.        7036310.
      2420740.98      7036073.55
#Sta/Elev= 30
  4209.8  524.31  4221.8   524.7  4241.8  519.11  4292.3  517.59  4398.3  517.19
  4482.4  516.85  4604.6  516.41  4807.4  514.88  4813.7  514.98  4819.3  516.89
  4853.9  518.32    4894   509.3  4924.1  500.49  4934.1  499.32  4954.2  499.76
  4964.2  497.36  4974.2  497.46  4984.3  500.99  4994.3  499.97  4994.5  497.36
    4996  496.86  5005.6  497.36  5006.9  499.08  5014.4  499.99  5024.4  505.17
  5044.4  511.62  5074.4  517.28  5094.9  518.12  5144.5  520.02  5241.1  521.46
#Mann= 9 ,-1 , 0
  4209.8    .075       0  4292.3      .1       0  4398.3    .075       0
  4482.4      .1       0  4604.6    .075       0  4807.4     .05       0
  4994.5     .05       0  5005.6     .05       0  5094.9      .1       0
Bank Sta=4994.5,5005.6
XS Rating Curve= 0 ,0
Exp/Cntr=0.3,0.1

Type RM Length L Ch R = 1 ,19547   ,261,261,261
BEGIN DESCRIPTION:
COTTONWOOD BR AT DENTON 29.0
END DESCRIPTION:
XS GIS Cut Line= 3
        2421061.      7036785.37      2421130.99      7036442.07
      2421104.47      7036173.54
#Sta/Elev= 30
  4625.3  517.89  4625.4  517.89  4722.6  516.86  4739.2  515.98  4753.2  513.81
  4789.7  513.12  4794.8  511.64  4834.9  512.94  4875.7  512.25  4885.7  509.53
  4890.8   509.3  4896.1  506.65  4916.5  501.11  4926.7  499.07  4941.4  498.18
  4947.2   495.6  4957.4  498.65  4967.6  498.61  4974.2  494.84  4979.2  494.84
  4987.8  496.88  4994.5  494.84    4996  494.34  5005.6  494.84  5007.9  497.53
    5028  500.81  5068.2  511.18  5128.5  517.33  5218.9  519.85  5245.5   522.2
#Mann= 4 ,-1 , 0
  4625.3    .075       0  4625.4     .05       0  4994.5    .033       0
  5005.6     .05       0
Bank Sta=4994.5,5005.6
XS Rating Curve= 0 ,0
Exp/Cntr=0.3,0.1

Type RM Length L Ch R = 1 ,19286   ,1172,1172,1172
BEGIN DESCRIPTION:
COTTONWOOD BR AT DENTON 28.5
END DESCRIPTION:
XS GIS Cut Line= 5
      2421210.99      7037041.93      2421384.28      7036608.71
      2421387.61       7036465.4      2421170.98      7036112.13
      2421104.32      7035658.85
#Sta/Elev= 30
  4344.3  514.73  4376.3  512.03  4393.1  511.72  4766.4  503.29  4963.8  504.57
  4972.3  502.07  4979.2  495.29  4994.5  494.54    4996  494.04  5005.6  494.54
  5007.5  499.95  5015.9  500.75  5052.7  499.13  5066.2  501.66    5190  501.25
    5248  502.81  5269.3   504.4  5277.3  504.17  5300.2  505.76  5321.5  508.25
  5327.3  515.47  5342.8  516.72  5348.6   518.4  5416.4  520.48    5584  522.53
  5695.4  524.26  5734.7  521.34  5760.1  521.41  5795.3  524.12  5826.8  524.41
#Mann= 6 ,-1 , 0
  4344.3     .05       0  4393.1     .12       0  4994.5     .07       0
  5005.6     .12       0  5269.3     .05       0    5584    .075       0
Bank Sta=4994.5,5005.6
XS Rating Curve= 0 ,0
Exp/Cntr=0.3,0.1

Type RM Length L Ch R = 1 ,18114   ,402,402,402
BEGIN DESCRIPTION:
COTTONWOOD BR AT DENTON 28.0
END DESCRIPTION:
XS GIS Cut Line= 4
      2421224.29      7037068.65      2421454.26      7036565.38
      2421550.91      7036175.45      2421943.12       7035623.7
#Sta/Elev= 30
  3942.2  515.84  3958.6  514.79  4041.5  510.72  4374.8  503.13  4614.2  503.56
  4686.5  500.58  4779.2  501.58  4810.1  498.34  4841.1  500.16  4992.4   499.8
  4994.5  488.24    4996  487.74  5005.6  488.24  5007.2  495.21    5022  488.24
  5028.1  490.65  5036.7  490.37  5042.9   495.9  5057.6  495.94  5072.4  499.68
  5158.5  502.36  5173.2  507.17  5179.4  511.77  5194.1  514.52  5200.3  518.89
  5238.3  523.13  5387.2  523.99    5402  520.72  5488.1  523.67  5574.2  523.07
#Mann= 5 ,-1 , 0
  3942.2     .05       0  3958.6     .12       0  4994.5     .07       0
  5005.6     .12       0  5238.3     .05       0
Bank Sta=4994.5,5005.6
XS Rating Curve= 0 ,0
Exp/Cntr=0.3,0.1

Type RM Length L Ch R = 1 ,17712   ,478,478,478
BEGIN DESCRIPTION:
COTTONWOOD BR AT DENTON 27.0
END DESCRIPTION:
XS GIS Cut Line= 4
      2421244.28      7037091.99      2421574.24      7036498.73
      2421867.35      7036424.71      2421967.51      7036045.47
#Sta/Elev= 30
  4212.8  516.39  4254.2  515.73  4313.7  510.79  4600.8  503.57  4725.4  501.99
  4812.3  503.85  4917.2  503.62  4927.5  501.75  4937.8  498.14  4945.3  497.31
  4968.8  498.38  4979.1  497.84  4986.4  489.56  4991.6  487.89  4994.5  487.89
    4996  487.39  5005.6  487.89    5010   494.8  5020.3  497.63  5073.6  502.32
  5082.2   504.6  5109.5  508.58  5114.7  508.04  5133.8  510.15  5150.6  517.15
  5164.7  518.62    5175  521.61  5355.9  522.84  5499.8  523.81  5586.2  523.41
#Mann= 5 ,-1 , 0
  4212.8     .12       0  4994.5     .07       0  5005.6     .12       0
  5355.9     .05       0  5499.8    .075       0
Bank Sta=4994.5,5005.6
XS Rating Curve= 0 ,0
Exp/Cntr=0.3,0.1

Type RM Length L Ch R = 1 ,17234   ,464,464,464
BEGIN DESCRIPTION:
COTTONWOOD BR AT DENTON 26.0
END DESCRIPTION:
XS GIS Cut Line= 3
      2421604.24      7037105.28        2421729.        7036910.
      2421940.28      7036363.55
#Sta/Elev= 30
  4773.3  516.56  4815.5  515.21  4851.9  509.36  4878.7  506.52  4924.7  502.87
  4939.9  502.98  4945.8   501.7  4955.1  488.69  4969.4  486.28  4982.2  491.02
  4991.5  492.75  4994.4  486.28    4996  485.78  5005.6  486.28  5007.7  495.85
  5014.6  497.16  5037.2  498.19  5049.9  496.74  5153.7  497.08  5165.8  496.03
  5230.2  497.88  5268.1  501.24  5401.7  506.52  5423.2  510.04  5431.7  512.66
    5437  512.67  5444.6  515.76  5455.3  517.81  5461.6  521.28  5590.9  522.49
#Mann= 4 ,-1 , 0
  4773.3     .05       0  4878.7     .12       0  4994.4     .07       0
  5005.6     .12       0
Bank Sta=4994.4,5005.6
XS Rating Curve= 0 ,0
Exp/Cntr=0.3,0.1

Type RM Length L Ch R = 1 ,16770   ,332,332,332
BEGIN DESCRIPTION:
COTTONWOOD BR AT DENTON 25.0
END DESCRIPTION:
XS GIS Cut Line= 4
       2421640.9      7037258.59      2422097.48      7036941.98
      2421960.84      7036448.74      2422113.72      7035833.89
#Sta/Elev= 30
  4240.4  518.32    4316  517.03  4337.6  516.36  4396.3  508.68  4506.1  505.24
  4712.7  499.96  4912.2  501.12  4953.7  496.19  4958.9  487.46  4974.5  493.16
  4993.2  492.55  4994.4  485.63  4995.9  485.13  5005.6  485.63  5026.4   486.5
  5037.9  492.51  5047.1     495  5140.5  497.75  5180.2  504.01  5185.4  503.06
  5202.8  506.93  5233.9  510.03  5259.2  515.66  5275.4   521.3  5442.2  523.36
  5659.7  523.36  5770.2  523.67  5812.1  521.35  5893.9  519.76  5941.4  522.04
#Mann= 9 ,-1 , 0
  4240.4     .05       0    4316     .12       0  4337.6     .05       0
  4506.1     .12       0  4994.4     .07       0  5005.6     .12       0
  5442.2     .05       0  5659.7    .075       0  5812.1     .05       0
Bank Sta=4994.4,5005.6
XS Rating Curve= 0 ,0
Exp/Cntr=0.3,0.1

Type RM Length L Ch R = 1 ,16438   ,610,610,610
BEGIN DESCRIPTION:
COTTONWOOD BR AT DENTON 24.0
END DESCRIPTION:
XS GIS Cut Line= 3
      2421610.92      7037308.57      2422317.44        7036832.
      2422794.04      7036498.72
#Sta/Elev= 30
  4196.1   519.4  4336.7  516.74  4366.1  514.56  4410.9  508.45  4770.7   499.1
  4812.7  500.87  4929.6  499.46  4950.6  493.98  4971.6  490.83  4977.8  485.31
  4986.6  484.54  4992.6  486.48  4994.4  484.54  4995.9  484.04  5005.6  484.54
  5007.6  491.81    5014  493.37  5052.3  492.88  5222.4  500.25  5309.7  507.15
  5317.4   508.7  5323.5  508.45  5338.4  511.94  5344.5  511.57  5353.2   514.2
  5367.5  515.33  5446.5  516.51  5517.1  519.29  5567.7  518.22  5629.9  521.25
#Mann= 6 ,-1 , 0
  4196.1     .05       0  4336.7     .12       0  4994.4     .07       0
  5005.6     .12       0  5309.7     .05       0  5446.5    .075       0
Bank Sta=4994.4,5005.6
XS Rating Curve= 0 ,0
Exp/Cntr=0.3,0.1

Type RM Length L Ch R = 1 ,15828   ,456,456,456
BEGIN DESCRIPTION:
COTTONWOOD BR AT DENTON 23.0
END DESCRIPTION:
XS GIS Cut Line= 4
      2421977.53      7037591.85      2422504.08      7037231.93
      2422650.72      7037198.61      2423000.67      7036958.64
#Sta/Elev= 30
  4336.2  514.14  4459.9  508.45  4489.7     502  4495.8  505.29  4501.9  503.99
  4525.6  496.66  4540.6   498.9  4546.6  495.74  4568.1  491.18  4612.3  488.79
  4929.3  492.02  4950.3  489.13  4979.1  489.51  4994.4  483.13  4995.9  482.63
  5005.7  483.13  5020.1  486.37  5030.3  491.66  5040.6  493.27  5061.1  493.13
  5071.3   495.8  5091.1  496.23  5112.4  499.12    5195  502.44  5207.4  504.92
  5241.1  504.44  5287.9  505.79  5352.7  512.93  5410.5  516.58  5548.7  516.81
#Mann= 5 ,-1 , 0
  4336.2     .05       0  4501.9     .12       0  4994.4     .07       0
  5005.7     .12       0  5241.1     .05       0
Bank Sta=4994.4,5005.7
XS Rating Curve= 0 ,0
Exp/Cntr=0.3,0.1

Type RM Length L Ch R = 1 ,15372   ,439,439,439
BEGIN DESCRIPTION:
COTTONWOOD BR AT DENTON 22.0
END DESCRIPTION:
XS GIS Cut Line= 3
      2422379.04      7037709.97      2422767.36      7037395.24
      2422920.65      7037235.28
#Sta/Elev= 30
  4466.8  503.75    4645  495.22  4651.4  497.03  4672.7  497.28  4708.9  492.03
  4729.7  493.17  4772.8  489.84  4779.3  491.47  4787.2  489.56    4808  489.57
  4828.8  492.99  4851.2  488.58    4872  488.02  4935.9  489.66  4950.3  491.73
  4956.7  487.73  4978.5  486.88  4985.8   481.4  4994.4   481.4  4995.9   480.9
  5005.7   481.4  5006.8  483.95  5014.1  488.69  5056.5  496.17  5063.5  500.54
  5077.6  502.92  5091.8  501.54  5115.8  507.37  5148.4  511.84  5188.2  513.36
#Mann= 4 ,-1 , 0
  4466.8     .12       0  4994.4     .07       0  5005.7     .12       0
  5115.8     .05       0
Bank Sta=4994.4,5005.7
XS Rating Curve= 0 ,0
Exp/Cntr=0.3,0.1

Type RM Length L Ch R = 1 ,14933   ,473,473,473
BEGIN DESCRIPTION:
COTTONWOOD BR AT DENTON 21.0
END DESCRIPTION:
XS GIS Cut Line= 3
      2422628.97      7037860.03        2422779.        7037710.
      2422979.02      7037559.99
#Sta/Elev= 30
  4783.1  500.53  4797.6  499.87  4797.8  499.86  4952.8  495.61  4991.7  485.44
  4994.4  480.14  4995.9  479.64  5005.7  480.14  5031.7  480.69    5038  483.14
  5052.6  481.39  5058.8  488.13  5067.2  485.47  5073.4  487.14  5102.6  489.11
  5108.8  490.36  5117.2  489.79  5123.4  491.51  5145.3  495.43  5158.8  495.75
  5167.2  496.94  5173.4  496.15  5181.7  498.62    5188   496.8  5202.6  499.11
  5208.8  498.89  5217.2  500.46    5238  500.85  5242.2  502.52  5245.3  502.52
#Mann= 5 ,-1 , 0
  4783.1     .12       0  4797.6     .05       0  4797.8     .12       0
  4994.4     .07       0  5005.7     .12       0
Bank Sta=4994.4,5005.7
XS Rating Curve= 0 ,0
Exp/Cntr=0.3,0.1

Type RM Length L Ch R = 1 ,14460   ,425,425,425
BEGIN DESCRIPTION:
COTTONWOOD BR AT DENTON 20.0
END DESCRIPTION:
XS GIS Cut Line= 3
      2422770.73      7038261.72        2423079.        7038010.
      2423267.25      7037845.18
#Sta/Elev= 30
  4602.5  517.44  4638.6  516.82  4645.1     512  4651.9  511.41  4659.5   514.1
  4665.9  509.94  4694.6  505.82  4702.5  506.04  4723.4  501.85  4740.8  502.45
  4808.1  502.83  4858.5  498.91  4900.7  492.27  4908.6  494.19    4915  491.85
    4923  494.49  4943.8  493.27  4972.5  486.28  4978.9  481.44  4994.4   478.6
  4995.9   478.1  5005.7   478.6  5007.6  482.31  5014.3  484.54  5050.3  487.72
  5085.4  493.92  5106.8  495.95  5113.9  494.74    5149  495.15  5250.7   501.2
#Mann= 4 ,-1 , 0
  4602.5     .05       0  4740.8     .12       0  4994.4     .07       0
  5005.7     .12       0
Bank Sta=4994.4,5005.7
XS Rating Curve= 0 ,0
Exp/Cntr=0.3,0.1

Type RM Length L Ch R = 1 ,14035   ,345,345,345
BEGIN DESCRIPTION:
COTTONWOOD BR AT DENTON 19.0
END DESCRIPTION:
XS GIS Cut Line= 3
      2423280.62      7038421.71      2423467.24      7038171.77
      2423477.24      7037895.18
#Sta/Elev= 30
  4625.9   510.5  4655.7  509.97  4697.5  510.24  4712.7  508.84  4776.8  504.96
    4783  502.95  4797.6  501.52  4847.8  493.11  4862.2  491.58  4903.9  491.36
  4926.9  487.74  4933.1  488.83  4935.8  487.51  4989.6  484.71  4994.3  477.74
  4995.9  477.24  5005.7  477.74  5009.6  484.19  5019.6  477.96  5029.7  477.74
  5039.7  483.63  5049.7  488.11  5069.7  489.78  5079.7   494.9  5099.7  494.18
  5119.7  495.23  5124.8  497.12  5129.8  496.42  5199.8  500.37  5214.6  500.36
#Mann= 6 ,-1 , 0
  4625.9     .05       0  4655.7     .12       0  4712.7     .05       0
  4847.8     .12       0  4994.3     .07       0  5005.7     .12       0
Bank Sta=4994.3,5005.7
XS Rating Curve= 0 ,0
Exp/Cntr=0.3,0.1

Type RM Length L Ch R = 1 ,13690   ,282,282,282
BEGIN DESCRIPTION:
COTTONWOOD BR AT DENTON 18.2
END DESCRIPTION:
XS GIS Cut Line= 4
      2423757.19      7038501.69      2423763.85      7038275.08
      2423747.19       7038175.1      2423753.84      7037493.39
#Sta/Elev= 30
  4730.8  504.06  4742.5  504.49  4792.5  495.31  4932.6   491.2  4952.5  487.03
  4957.5  487.03  4962.7  482.12  4972.8  478.66  4982.9   477.6  4994.3  477.49
  4995.9  476.99  5005.7  477.49  5012.9  483.58    5025  485.75    5084  485.62
    5114  487.31    5144   487.1    5154  487.94    5174  491.18    5194  490.73
    5234  491.55    5264  491.31    5344   493.4    5404  493.92    5414  494.88
    5424  494.28    5494  497.41    5554  497.86  5626.5  500.99  5740.6  506.69
#Mann= 5 ,-1 , 0
  4730.8     .05       0  4994.3    .033       0  5005.7     .05       0
    5025     .12       0  5626.5     .05       0
Bank Sta=4994.3,5005.7
XS Rating Curve= 0 ,0
Exp/Cntr=0.3,0.1

Type RM Length L Ch R = 1 ,13408   ,319,319,319
BEGIN DESCRIPTION:
COTTONWOOD BR AT DENTON 18.0
END DESCRIPTION:
XS GIS Cut Line= 3
      2423957.15       7038511.7      2423953.82      7038015.13
      2423963.82      7037555.22
#Sta/Elev= 30
  4548.4  503.21  4740.1  497.36  4810.1  496.59  4820.1  494.67  4920.1  494.66
  4930.1  494.29  4938.9  492.27  4950.1  486.77  4960.1  485.14  4980.1  485.03
  4994.3  476.14  4995.9  475.64  5005.7  476.14  5010.1   476.3  5021.7  482.32
  5030.1   485.1    5040  485.85  5049.2  486.47  5070.1  484.84  5080.1  485.71
  5090.1  489.31  5150.1   489.8  5240.2  492.49  5260.2  496.58  5300.2  496.34
  5320.2  497.42  5350.2  502.77  5400.2  504.69  5410.2  507.83    5505  511.25
#Mann= 4 ,-1 , 0
  4548.4     .05       0  4938.9     .12       0  4994.3     .07       0
  5005.7     .12       0
Bank Sta=4994.3,5005.7
XS Rating Curve= 0 ,0
Exp/Cntr=0.3,0.1

Type RM Length L Ch R = 1 ,13089   ,360,360,360
BEGIN DESCRIPTION:
COTTONWOOD BR AT DENTON 17.0
END DESCRIPTION:
XS GIS Cut Line= 3
      2424053.79      7038471.76      2424210.44      7037955.14
      2424110.85      7037553.45
#Sta/Elev= 30
  4413.7  499.54  4521.5  495.26  4685.1  496.19  4795.2  495.33  4822.9  493.39
  4828.1  490.55  4854.4  490.86  4885.8  487.53  4917.1  486.45  4932.1  487.53
  4969.1  481.58  4977.3  476.35  4982.5  474.99  4989.8  475.82  4994.3  474.99
  4995.9  474.49  5005.7  474.99  5010.4  487.02  5082.5  490.05  5113.4  492.98
    5177  496.57  5230.8  497.57    5237  500.04  5242.2  500.58  5272.1  503.42
  5298.8  504.35  5313.5  503.76  5319.4  502.12    5340  504.89  5367.4  505.62
#Mann= 6 ,-1 , 0
  4413.7     .05       0  4685.1     .12       0  4994.3     .07       0
  5005.7     .12       0    5177     .05       0  5242.2     .12       0
Bank Sta=4994.3,5005.7
XS Rating Curve= 0 ,0
Exp/Cntr=0.3,0.1

Type RM Length L Ch R = 1 ,12729   ,426,426,426
BEGIN DESCRIPTION:
COTTONWOOD BR AT DENTON 16.0
END DESCRIPTION:
XS GIS Cut Line= 3
      2424628.99      7038359.98        2424529.        7038010.
      2424479.01      7037760.03
#Sta/Elev= 30
  4631.2  503.28  4641.6  502.94  4653.3  500.78  4662.4  496.07  4681.9  494.82
    4704  494.88  4754.7  497.44  4825.4  496.87  4832.7  496.64  4839.2  493.15
  4849.6  490.42  4922.4  486.59  4973.1  485.77  4984.8  484.66  4992.6  484.79
  4994.3  473.83  4995.8  473.33  5004.2  473.33  5005.8  473.83  5015.6  473.83
  5025.8  474.61    5036  481.14  5046.2  483.89  5066.6  485.56  5117.6  485.92
  5129.8   487.5  5148.2  489.93  5178.7  492.77  5209.3  500.26  5250.1  501.45
#Mann= 5 ,-1 , 0
  4631.2    .075       0  4825.4     .12       0  4994.3     .07       0
  5005.8     .12       0  5129.8    .075       0
Bank Sta=4994.3,5005.8
XS Rating Curve= 0 ,0
Exp/Cntr=0.3,0.1

Type RM Length L Ch R = 1 ,12303   ,466,466,466
BEGIN DESCRIPTION:
COTTONWOOD BR AT DENTON 15.0
END DESCRIPTION:
XS GIS Cut Line= 3
      2424893.65      7038438.37        2424879.        7037960.
      2424829.01      7037660.03
#Sta/Elev= 30
  4522.2  502.74  4526.3  502.83  4560.6  502.75  4590.6  495.71  4600.6  494.97
  4620.6  495.02  4670.6  497.06  4750.7  495.87  4760.7  494.98  4770.7  489.87
  4810.7  486.92  4877.7  485.26  4940.8   484.1  4980.8  484.82  4990.8  483.52
  4994.2  472.89  4995.8  472.39  5005.8  472.89  5010.9  476.18  5021.1  472.92
  5028.7  472.89  5041.3  479.93  5051.5  482.66  5089.5  486.46  5094.6   486.3
  5150.3  491.59  5155.4  491.56  5173.1  493.98  5277.1   501.6  5304.9   504.4
#Mann= 5 ,-1 , 0
  4522.2    .075       0  4526.3     .05       0  4877.7     .12       0
  4994.2     .07       0  5005.8     .12       0
Bank Sta=4994.2,5005.8
XS Rating Curve= 0 ,0
Exp/Cntr=0.3,0.1

Type RM Length L Ch R = 1 ,11837   ,417,417,417
BEGIN DESCRIPTION:
COTTONWOOD BR AT DENTON 14.0
END DESCRIPTION:
XS GIS Cut Line= 3
       2425110.3      7038455.01        2425279.        7038060.
      2425416.89      7037785.18
#Sta/Elev= 30
  4565.9  501.46  4576.1   499.3  4605.1  495.55  4669.2   496.8  4728.6  496.12
  4745.3  492.74  4749.6  490.75  4752.2  489.54  4799.4   485.7    4852  483.34
  4897.6  482.54  4960.1  483.02  4986.3   482.5  4992.7  476.32  4994.2   472.1
  4995.8   471.6  5005.9   472.1  5017.8   472.1  5026.1  477.79  5031.7  484.51
  5040.2  486.83  5062.6  489.53  5084.9  490.42  5098.7  492.17  5143.4  495.96
  5188.1   498.8  5196.8  500.43  5232.8  504.27  5277.4  505.85  5302.9   505.4
#Mann= 5 ,-1 , 0
  4565.9    .075       0  4749.6     .05       0  4960.1     .12       0
  4994.2     .07       0  5005.9     .12       0
Bank Sta=4994.2,5005.9
XS Rating Curve= 0 ,0
Exp/Cntr=0.3,0.1

Type RM Length L Ch R = 1 ,11420   ,469,469,469
BEGIN DESCRIPTION:
COTTONWOOD BR AT DENTON 13.0
END DESCRIPTION:
XS GIS Cut Line= 3
       2425173.6      7038491.71        2425529.        7038360.
      2425870.17      7038168.42
#Sta/Elev= 30
    4625  500.27  4645.5  498.22  4662.8   494.5  4675.9  493.63    4701  493.49
  4756.4  495.39  4811.8  494.82  4817.2  491.98  4822.7  487.47  4840.1  485.96
  4872.6  482.97    4903   481.8  4988.8  481.47  4994.2  472.56  4995.8  472.06
  5005.9  472.56  5017.7  472.84  5033.7  482.02  5107.2  484.23  5120.4  490.89
    5156  492.37    5255  490.73  5267.8  491.49  5271.2  492.85  5276.6  495.01
  5290.7  498.61  5341.7  498.78  5369.3  500.91  5379.3  501.21  5395.3  503.18
#Mann= 7 ,-1 , 0
    4625    .075       0  4840.1     .12       0  4994.2     .07       0
  5005.9     .12       0    5156     .05       0  5271.2    .075       0
  5369.3     .05       0
Bank Sta=4994.2,5005.9
XS Rating Curve= 0 ,0
Exp/Cntr=0.3,0.1

Type RM Length L Ch R = 1 ,10951   ,416,416,416
BEGIN DESCRIPTION:
COTTONWOOD BR AT DENTON 12.0
END DESCRIPTION:
XS GIS Cut Line= 3
      2425203.57      7038858.32        2425629.        7038760.
      2425960.15      7038628.35
#Sta/Elev= 30
  4568.3  501.53  4594.4  500.98  4604.7  496.78  4634.9  497.26  4676.7  497.25
  4707.3  495.75  4748.4  496.03  4779.1  493.41  4789.4  487.73  4804.9  484.19
  4851.2  482.91  4943.4   481.2  4974.2  479.21  4986.1  472.48  4994.2  470.57
  4995.8  470.07  5005.9  470.57  5014.4  476.94  5026.5  480.96  5049.5  479.87
    5091  480.11  5127.7  482.85  5134.1  485.19  5144.8  486.45    5152  488.35
  5166.4  494.62    5190  494.75  5220.2  494.13    5260  495.02  5361.3  499.62
#Mann= 6 ,-1 , 0
  4568.3    .075       0  4634.9     .05       0  4851.2     .12       0
  4994.2     .07       0  5005.9     .12       0    5190     .05       0
Bank Sta=4994.2,5005.9
XS Rating Curve= 0 ,0
Exp/Cntr=0.3,0.1

Type RM Length L Ch R = 1 ,10535   ,292,292,292
BEGIN DESCRIPTION:
COTTONWOOD BR AT DENTON 11.0
END DESCRIPTION:
XS GIS Cut Line= 3
      2425350.23      7039291.57        2425829.        7039060.
       2426140.1      7038778.33
#Sta/Elev= 30
  4468.2  496.68  4493.1  496.36  4528.6  495.23  4534.1     496  4573.8  490.48
  4624.5   490.2  4664.1  487.29  4731.9  487.63  4737.5  487.26  4744.5  484.89
    4760  485.19  4777.1  484.25    4789  479.84  4804.8  479.37  4895.6  477.89
  4963.4  479.75  4968.9   479.2  4977.8  472.24  4994.2  470.32  4995.8  469.82
  5005.9  470.32  5021.3  479.08  5056.5  480.57  5078.1  479.01  5120.7   479.2
  5205.1   484.4  5247.7  488.67  5290.3  491.63  5397.4  497.03  5419.7  497.41
#Mann= 6 ,-1 , 0
  4468.2     .05       0  4493.1    .075       0  4804.8     .12       0
  4994.2     .07       0  5005.9     .12       0  5397.4     .05       0
Bank Sta=4994.2,5005.9
XS Rating Curve= 0 ,0
Exp/Cntr=0.3,0.1

Type RM Length L Ch R = 1 ,10243   ,183,183,183
BEGIN DESCRIPTION:
COTTONWOOD BR AT DENTON 10.2
END DESCRIPTION:
XS GIS Cut Line= 3
      2425422.37      7039596.68      2425922.35      7039346.69
      2426699.97      7038655.04
#Sta/Elev= 30
    4375  503.68  4388.9   502.3  4491.8  502.07  4527.8  497.83    4579  498.78
  4623.8  490.24  4735.6  489.28    4833   476.2  4957.3  478.22  4971.5  477.06
    4979  468.86  4994.2  468.86  4995.8  468.36  5005.9  468.86  5007.4  475.17
  5028.4  477.92  5248.3  479.02  5297.6  482.04  5332.7  488.46  5389.6  483.99
  5517.5   488.5  5524.2  485.69  5531.7  488.08  5538.4  484.28  5545.1  488.94
  5609.5  487.54  5758.3  497.61    5843  497.24  5920.6  495.59  5974.7  499.69
#Mann= 7 ,-1 , 0
    4375    .075       0  4388.9     .05       0  4491.8    .075       0
    4833     .05       0  4994.2    .033       0  5005.9     .05       0
    5843    .075       0
Bank Sta=4994.2,5005.9
XS Rating Curve= 0 ,0
Exp/Cntr=0.3,0.1

Type RM Length L Ch R = 1 ,10060   ,441,441,441
BEGIN DESCRIPTION:
COTTONWOOD BR AT DENTON 10.0
END DESCRIPTION:
XS GIS Cut Line= 3
      2425528.99        7039710.        2426029.        7039460.
      2426628.96      7038960.03
#Sta/Elev= 30
  4447.9  506.72  4662.3  491.88  4702.3  487.33    4782  483.29  4872.8  478.75
  4894.1  473.72  4917.5  477.32  4939.8  477.49  4948.2  475.82  4953.8  476.84
  4962.2   470.8  4970.6  469.04  4984.6  468.44  4992.9  471.62  4994.1  468.44
  4995.7  467.94    5006  468.44  5006.9  477.64  5014.1  479.62  5020.6  478.98
  5028.4  474.26  5042.7  473.37  5123.6  474.38  5254.9  477.08  5575.1  489.02
  5681.9  490.38  5745.6  495.52  5752.2  494.35  5766.5  497.55  5787.9  499.24
#Mann= 7 ,-1 , 0
  4447.9     .05       0  4662.3    .075       0    4782     .05       0
  4894.1     .12       0  4994.1     .07       0    5006     .12       0
  5123.6     .05       0
Bank Sta=4994.1,5006
XS Rating Curve= 0 ,0
Exp/Cntr=0.3,0.1

Type RM Length L Ch R = 1 ,9619    ,472,472,472
BEGIN DESCRIPTION:
COTTONWOOD BR AT DENTON 9.0
END DESCRIPTION:
XS GIS Cut Line= 3
      2425629.04        7039810.        2426079.        7039860.
      2426629.03      7039409.97
#Sta/Elev= 30
  4542.5  500.03  4562.6  499.39  4602.8  490.61  4643.1  487.86  4663.2  485.59
  4733.6  483.98  4773.9  480.37  4814.1  480.54  4894.6  478.93  4934.5  476.01
    4965   475.9  4985.2  468.89  4994.1  468.51  4995.7  468.01    5006  468.51
  5008.9  475.88  5016.8  476.56  5023.2  474.53  5031.1  473.34    5046   473.3
  5130.2   474.7  5251.5  472.71  5393.6   474.1  5449.6  476.87  5486.2  481.63
  5513.5  484.11  5577.4  484.99  5649.2  491.79  5684.3  493.73  5705.9  496.13
#Mann= 5 ,-1 , 0
  4542.5     .05       0  4934.5     .12       0  4994.1     .07       0
    5006     .12       0    5046     .05       0
Bank Sta=4994.1,5006
XS Rating Curve= 0 ,0
Exp/Cntr=0.3,0.1

Type RM Length L Ch R = 1 ,9147    ,374,374,374
BEGIN DESCRIPTION:
COTTONWOOD BR AT DENTON 8.0
END DESCRIPTION:
XS GIS Cut Line= 3
      2425633.53      7040304.72      2426190.09       7040261.4
      2427129.95      7039691.48
#Sta/Elev= 30
  4501.2  482.76  4586.9  481.28  4647.1  481.89  4727.3   479.8  4767.5  479.85
  4797.6  478.16  4897.9   477.2    4958  474.16  4968.1  471.65  4978.1  465.84
  4994.1  465.81  4995.7  465.31    5006  465.81  5008.1  474.49  5013.1  473.43
  5018.2  474.57  5038.3  472.79  5106.7  473.22  5269.6  472.35  5306.4   471.1
  5321.9  468.35  5395.6  468.43  5432.4     472  5701.4  475.61  5839.6  482.24
  5998.6  482.07  6014.1  483.23  6078.1  483.67  6114.9  485.47  6158.6  485.67
#Mann= 4 ,-1 , 0
  4501.2     .05       0  4994.1     .05       0    5006     .05       0
  5106.7     .05       0
Bank Sta=4994.1,5006
XS Rating Curve= 0 ,0
Exp/Cntr=0.3,0.1

Type RM Length L Ch R = 1 ,8773    ,892,892,892
BEGIN DESCRIPTION:
COTTONWOOD BR AT DENTON 7.6
END DESCRIPTION:
XS GIS Cut Line= 3
      2425733.52      7040957.93      2426356.73      7040524.68
      2427249.88      7039878.15
#Sta/Elev= 30
  4358.7  479.93  4561.4  479.09  4626.9  477.81  4718.2  478.11  4835.6   475.2
    4922  475.97  4942.9  472.84  4957.6  473.29  4978.7  473.37  4993.6  465.55
  4994.1  464.42  4995.7  463.92    5006  464.42  5008.4  470.67  5014.5  473.71
    5023  473.95  5029.3  472.42  5109.7  472.02  5358.6  469.56  5559.7  470.51
  5624.6  471.17  5716.6  474.43  5731.3  475.55  5737.8  477.49    5746  478.35
  5774.8  479.16    5811  482.41    5968  481.89    6060  482.84  6220.3  481.37
#Mann= 6 ,-1 , 0
  4358.7    .075       0  4718.2     .05       0  4957.6     .12       0
  4994.1     .07       0    5006     .12       0  5109.7     .05       0
Bank Sta=4994.1,5006
XS Rating Curve= 0 ,0
Exp/Cntr=0.3,0.1

Type RM Length L Ch R = 1 ,7881    ,589,589,589
BEGIN DESCRIPTION:
COTTONWOOD BR AT DENTON 7.2
END DESCRIPTION:
XS GIS Cut Line= 3
      2426076.76       7041217.9      2426792.38      7041040.07
      2427645.25      7040369.03
#Sta/Elev= 30
  4052.5  479.14  4237.4  477.36  4580.3  473.81  4599.7  473.28  4611.2  470.23
  4621.5  469.13  4675.9  469.14  4809.5  468.68  4904.1  470.08    4973  471.29
  4987.5  468.33    4994  462.75  4995.7  462.25    5006  462.75  5008.3  462.75
  5014.7  469.14  5022.7   470.6  5032.9  470.09  5086.9  469.34    5143  466.73
  5210.9  468.16    5290  468.52  5349.9  469.78  5385.1  472.83  5449.3  475.81
  5585.7  476.31  5620.9  478.58    5799  479.55  5813.4  481.53  5875.1  482.04
#Mann= 9 ,-1 , 0
  4052.5     .05       0  4237.4    .075       0  4675.9     .05       0
  4904.1     .12       0    4994     .07       0    5006     .12       0
  5032.9     .05       0  5210.9     .12       0    5290     .05       0
Bank Sta=4994,5006
XS Rating Curve= 0 ,0
Exp/Cntr=0.3,0.1

Type RM Length L Ch R = 1 ,7292    ,450,450,450
BEGIN DESCRIPTION:
COTTONWOOD BR AT DENTON 7.0
END DESCRIPTION:
XS GIS Cut Line= 3
      2426112.65      7041562.52        2427079.        7041410.
      2428030.84      7040641.77
#Sta/Elev= 30
  4021.4  479.62  4239.4  479.97  4321.3   474.8  4469.1  476.57  4706.1  474.16
  4726.4  472.74  4773.6  473.99  4797.2  472.57  4807.4  468.98  4827.8  469.65
  4979.5  469.37  4989.6   468.9    4994  462.15  4995.7  461.65    5006  462.15
  5013.3  463.53  5027.7  469.46  5057.5  468.67  5134.9  466.63  5405.1  466.01
  5497.9  468.08  5646.6   474.8  5788.9  477.79  5824.1  481.08  5860.7  474.92
    6088  474.05  6108.8  472.87  6137.6  474.55  6172.8  478.73  6222.9  478.72
#Mann= 7 ,-1 , 0
  4021.4    .075       0  4239.4     .05       0  4469.1    .075       0
  4827.8     .12       0    4994     .07       0    5006     .12       0
  5057.5     .05       0
Bank Sta=4994,5006
XS Rating Curve= 0 ,0
Exp/Cntr=0.3,0.1

Type RM Length L Ch R = 1 ,6842    ,570,570,570
BEGIN DESCRIPTION:
COTTONWOOD BR AT DENTON 6.0
END DESCRIPTION:
XS GIS Cut Line= 3
      2426903.29      7042051.09      2427283.23      7041777.79
      2428043.12      7041201.21
#Sta/Elev= 30
  4558.8  472.69  4578.2  472.61    4614  474.76  4713.7  474.71  4771.9  473.23
  4878.7  473.94  4895.7  471.66  4935.4  468.23  4985.5  468.24    4994  459.54
  4995.7  459.04    5006  459.54  5008.8  468.19    5015  464.98  5021.1  459.54
  5026.8  459.54  5044.2  468.71  5052.1  468.74  5101.7  467.27  5121.9  467.33
  5135.7  465.52    5144  466.91  5158.6  467.11  5258.4  464.97    5502  464.87
  5564.2  465.18  5572.5     467  5614.1  468.35    5792  469.79  5980.7  473.25
#Mann= 9 ,-1 , 0
  4558.8     .05       0    4614    .075       0  4895.7     .05       0
    4994     .05       0    5006     .05       0  5052.1     .12       0
  5101.7     .05       0    5502    .075       0    5792      .1       0
Bank Sta=4994,5006
XS Rating Curve= 0 ,0
Exp/Cntr=0.3,0.1

Type RM Length L Ch R = 1 ,6272    ,496,496,496
BEGIN DESCRIPTION:
COTTONWOOD BR AT DENTON 5.0
END DESCRIPTION:
XS GIS Cut Line= 3
       2427269.9      7042577.66      2427583.18      7042141.06
      2428073.07      7041401.22
#Sta/Elev= 30
  4443.8  474.47  4570.5  474.06    4600   475.5  4656.5  475.48  4677.4  474.85
    4713  471.84  4792.8  473.86  4834.8   473.8    4864  471.36  4871.7  466.51
  4902.7  465.62  4964.7  466.26  4978.7  458.73    4994  458.72  4995.7  458.22
    5006  458.72  5006.6  464.88  5015.7  465.48  5021.7  464.72  5036.7  466.93
    5124  466.63    5151  465.06  5217.2  464.93  5232.3  462.51    5285  464.74
  5304.3  465.91  5486.2  467.84    5512  468.52  5642.1  467.72  5868.5  471.59
#Mann= 7 ,-1 , 0
  4443.8    .075       0  4902.7     .12       0    4994     .07       0
    5006     .12       0    5285     .05       0  5304.3    .075       0
  5486.2      .1       0
Bank Sta=4994,5006
XS Rating Curve= 0 ,0
Exp/Cntr=0.3,0.1
