--- Cade Branch.prj (project) ---

Proj Title=Cade Branch Base Level Engineering
Current Plan=p01
Default Exp/Contr=0.3,0.1
English Units
Geom File=g01
Flow File=f01
Plan File=p01
Y Axis Title=Elevation
X Axis Title(PF)=Main Channel Distance
X Axis Title(XS)=Station
BEGIN DESCRIPTION:
Cade Branch
END DESCRIPTION:
DSS Export Rating Curves= 0
DSS Export Rating Curve Sorted= 0
DSS Export Volume Flow Curves= 0
DXF OffsetX= 0
DXF OffsetY= 0
DXF ScaleX= 1
DXF ScaleY= 10

--- Cade Branch.p01 (plan) ---

Plan Title=Multiple Run
Program Version=4.10
Short Identifier=Multiple
Geom File=g01
Flow File=f01
Subcritical Flow
K Sum by GR= 0
Std Step Tol= 0.01
Critical Tol= 0.01
Num of Std Step Trials= 20
Max Error Tol= 0.3
Flow Tol Ratio= 0.001
Split Flow NTrial= 30
Split Flow Tol= 0.02
Split Flow Ratio= 0.02
Log Output Level= 0
Friction Slope Method= 1
Unsteady Friction Slope Method= 2
Unsteady Bridges Friction Slope Method= 1
Parabolic Critical Depth
Global Vel Dist= 1 , 1 , 1
Global Log Level= 0
CheckData=True
Encroach Param=-1 ,0,0, 0
BEGIN DESCRIPTION:
Multiple Run
END DESCRIPTION:
Computation Interval=1HOUR
Output Interval=1HOUR
Run HTab= 0
Run UNet= 0
Run PostProcess= 0
Run WQNet= 0
UNET Theta= 1
UNET Theta Warmup= 1
UNET ZTol= 0.02
UNET ZSATol= 0.05
UNET MxIter= 20
UNET MaxInSteps= 0
UNET DtIC= 0
UNET DtMin= 0
UNET MaxCRTS= 20
UNET WFStab= 2
UNET SFStab= 1
UNET WFX= 1
UNET SFX= 1
UNET DSS MLevel= 4
UNET DZMax Abort= 100
UNET Convert EG Bridges= 0
UNET Use Existing IB Tables=-1
UNET Froude Reduction=False
UNET Froude Limit= 1
UNET Froude Power= 10
UNET Time Slicing=0,0, 5
UNET Junction Losses=0
Instantaneous Interval=1HOUR
Write IC File= 0
Write IC File at Sim End=0
Echo Input=False
Echo Parameters=False
Echo Output=False
Write Detailed= 0
WQ AD Non Conservative
WQ ULTIMATE=-1
WQ Max Comp Step=1HOUR
WQ Output Interval=15MIN
WQ Output Selected Increments= 0
WQ Output face flow=0
WQ Output face velocity=0
WQ Output face area=0
WQ Output face dispersion=0
WQ Output cell volume=0
WQ Output cell surface area=0
WQ Output cell continuity=0
WQ Output cumulative cell continuity=0
WQ Output face conc=0
WQ Output face dconc_dx=0
WQ Output face courant=0
WQ Output face peclet=0
WQ Output face adv mass=0
WQ Output face disp mass=0
WQ Output cell mass=0
WQ Output cell source sink temp=0
WQ Output cell source sink nsm=0
WQ Output MaxMinRange=-1
WQ Daily Max Min Mean=-1
WQ Daily Range=0
WQ Daily Time=0
WQ Create Restart=0
WQ Fixed Restart=0
WQ System Summary=0
WQ Use Fixed Temperature=0
Sorting and Armoring Iterations= 10
XS Update Threshold= 0.02
Hydraulics Update Threshold= 0.02
Energy Slope Method= 1
Volume Change Method= 0
XS Weighting Method= 0
Number of US Weighted Cross Sections= 1
Number of DS Weighted Cross Sections= 1
Upstream XS Weight=0.25
Main XS Weight=0.5
Downstream XS Weight=0.25
Number of DS XS's Weighted with US Boundary= 1
Upstream Boundary Weight= 1
Weight of XSs Associated with US Boundary= 0
Number of US XS's Weighted with DS Boundary= 1
Downstream Boundary Weight= 0.5
Weight of XSs Associated with DS Boundary= 0.5
Sediment Output Level= 4
Mass or Volume Output= 0
Output Increment Type= 1
Profile and TS Output Increment= 10
XS Output Flag= 0
XS Output Increment= 10
Disregard all LS=0
Disregard all Conn=0
Disregard all Breaches=0
Disregard all Pumps=0

--- Cade Branch.f01 (steady flow) ---

Flow Title=Multiple
Number of Profiles=7
Profile Names=10-year,25-year,50-year,1pct_min,100-year,1pct_plu,500-year
River Rch & RM= Cade Branch,Reach-1,18248
     411     541     643     380     758    1512    1050
River Rch & RM= Cade Branch,Reach-1,17600
     586     788     951     569    1135    2264    1614
River Rch & RM= Cade Branch,Reach-1,14270
     652     888    1081     653    1302    2599    1895
River Rch & RM= Cade Branch,Reach-1,11717
     801    1103    1353     823    1641    3275    2421
River Rch & RM= Cade Branch,Reach-1,7756
     974    1356    1675    1025    2046    4082    3059
River Rch & RM= Cade Branch,Reach-1,2872
    1129    1586    1972    1214    2422    4833    3665
Boundary for River Rch & Prof#=Cade Branch,Reach-1,1
Up Type=0
Dn Type=3
Dn Slope=0.005
Boundary for River Rch & Prof#=Cade Branch,Reach-1,2
Up Type=0
Dn Type=3
Dn Slope=0.005
Boundary for River Rch & Prof#=Cade Branch,Reach-1,3
Up Type=0
Dn Type=3
Dn Slope=0.005
Boundary for River Rch & Prof#=Cade Branch,Reach-1,4
Up Type=0
Dn Type=3
Dn Slope=0.005
Boundary for River Rch & Prof#=Cade Branch,Reach-1,5
Up Type=0
Dn Type=3
Dn Slope=0.005
Boundary for River Rch & Prof#=Cade Branch,Reach-1,6
Up Type=0
Dn Type=3
Dn Slope=0.005
Boundary for River Rch & Prof#=Cade Branch,Reach-1,7
Up Type=0
Dn Type=3
Dn Slope=0.005

--- Cade Branch.g01 (geometry) ---

Geom Title=Existing Conditions
Program Version=4.10

River Reach=Cade Branch     ,Reach-1
Reach XY= 30
        2356029.        7048010.      2356285.21       7048017.8
      2356773.61      7048507.56        2356737.      7048913.33
      2357725.86      7050761.64      2357642.52      7050973.44
      2358271.16      7051112.93      2358186.52      7051356.93
      2358652.85      7051382.25      2358929.05      7051775.34
       2358736.2      7052116.08      2359373.42      7052315.58
      2359825.17      7053061.58      2359736.59      7053709.99
      2359877.97      7054149.57      2359579.18      7054444.91
        2359729.       7054552.5      2359973.81      7054414.56
      2360078.03      7055049.75       2359827.3       7055356.7
      2359428.56      7055380.03      2359778.02      7055670.26
      2359631.49      7056401.85      2360071.24      7056606.58
      2359737.83      7057053.06      2359880.04      7057225.18
      2359730.18      7057449.49      2360223.67      7057657.34
      2360182.54      7058108.53        2360879.        7059460.

Type RM Length L Ch R = 1 ,18248   ,133,133,133
BEGIN DESCRIPTION:
Cade Branch 39.0
END DESCRIPTION:
XS GIS Cut Line= 3
      2355967.81      7048510.07      2356076.33      7048082.52
      2356094.45      7047596.87
#Sta/Elev= 30
  4486.3  661.47  4610.2  660.94  4634.7  659.11  4651.4  654.51  4661.8  652.63
  4682.4   651.2  4793.4  650.44  4857.8  651.83  4899.1  651.32  4909.4  651.77
  4916.2  653.27  4931.2  653.35  4939.9  652.12  4949.9  651.65    4980  651.21
    4990  647.83    4998  646.14  4998.2  645.64  5001.7  645.64    5002  646.14
    5050  646.41    5070  651.27    5080  652.04  5110.1  651.92  5134.1  650.66
  5160.1  651.87  5200.1   651.6  5260.2  652.46  5340.2  652.57  5413.4  654.52
#Mann= 3 ,-1 , 0
  4486.3     .05       0    4998     .05       0    5002     .05       0
Bank Sta=4998,5002
XS Rating Curve= 0 ,0
Exp/Cntr=0.3,0.1

Type RM Length L Ch R = 1 ,18115   ,198,198,198
BEGIN DESCRIPTION:
Cade Branch 38.0
END DESCRIPTION:
XS GIS Cut Line= 3
      2355998.18       7048501.4      2356210.88      7048045.63
        2356229.      7047560.03
#Sta/Elev= 30
  4461.1  659.65  4471.5  660.47    4477  656.15  4494.4   658.2  4499.9  654.68
  4517.2  656.74  4522.7  653.48  4545.6  656.15  4551.1  652.35  4568.5  653.73
    4574  651.89  4591.3  652.35    4637  651.43  4793.7  652.29    4905   651.3
  4915.1  651.53  4922.4  652.75  4964.1  650.07  4969.7  647.28  4979.7  644.45
  4987.7  644.08    4988  643.58  4991.7  644.08  5009.7  645.12  5046.3  651.73
  5119.8  651.05  5149.8  652.66  5320.4  653.56  5378.1  654.76    5450  655.91
#Mann= 4 ,-1 , 0
  4461.1     .05       0  4987.7     .05       0  4991.7     .05       0
  5378.1    .075       0
Bank Sta=4987.7,4991.7
XS Rating Curve= 0 ,0
Exp/Cntr=0.3,0.1

Type RM Length L Ch R = 1 ,17917   ,317,317,317
BEGIN DESCRIPTION:
Cade Branch 37.0
END DESCRIPTION:
XS GIS Cut Line= 4
      2356137.09      7048828.64      2356206.46      7048292.94
       2356347.6      7048118.98      2356715.25      7047915.69
#Sta/Elev= 30
  4208.1  654.66    4257  653.75    4262  654.31  4277.3  653.47  4307.6  654.35
  4368.1  653.26  4429.9   654.4  4458.8  653.72  4499.8  650.89  4519.3  646.32
  4529.4  642.95  4539.5  638.35  4759.4  639.58  4837.7  638.27  4858.5  636.97
  4906.3  636.15  5017.9  637.11  5023.6  638.32  5088.9  640.21  5120.9     644
  5126.7  643.39  5142.7  646.76  5148.4  645.95  5164.5  648.38    5208  649.16
  5311.1  648.56  5332.8  650.59  5348.9  650.09  5354.6  651.97  5392.4  651.89
#Mann= 4 ,-1 , 0
  4208.1    .075       0  4429.9     .05       0  4858.5    .035       0
  5017.9     .05       0
Bank Sta=4858.5,5017.9
XS Rating Curve= 0 ,0
Exp/Cntr=0.3,0.1

Type RM Length L Ch R = 1 ,17600   ,323,323,323
BEGIN DESCRIPTION:
Cade Branch 36.0
END DESCRIPTION:
XS GIS Cut Line= 3
      2356176.16      7048934.94      2356436.57      7048448.84
      2356894.24      7047921.77
#Sta/Elev= 30
  4356.4  653.42  4397.1  654.26  4410.7  654.63  4458.1  655.47  4474.3   654.4
  4577.6  652.48  4600.2  653.21  4605.9  652.05  4627.9  651.56    4657  653.09
  4702.3  651.35  4721.4  652.19  4737.5  652.96  4804.4  650.96  4813.9  648.31
  4819.6  648.64  4835.8  644.24  4841.5  644.54  4849.8  641.15  4857.8   639.2
  4901.6  637.18  5027.3  636.18  5227.5  636.94  5270.3  637.92  5284.5  642.45
  5291.1  642.76  5298.8  644.83    5313  646.64  5546.6  647.57  5605.9  650.74
#Mann= 6 ,-1 , 0
  4356.4    .075       0  4397.1      .1       0  4410.7    .075       0
  4721.4     .05       0  4901.6    .033       0  5227.5     .05       0
Bank Sta=4901.6,5227.5
XS Rating Curve= 0 ,0
Exp/Cntr=0.3,0.1

Type RM Length L Ch R = 1 ,17277   ,412,412,412
BEGIN DESCRIPTION:
Cade Branch 35.0
END DESCRIPTION:
XS GIS Cut Line= 3
      2356440.92      7048772.18      2356781.63      7048464.03
      2357204.37      7048056.47
#Sta/Elev= 30
  4574.5  653.19  4645.5  652.92  4659.6  652.38  4666.4  650.04  4673.8  649.94
  4801.8  650.61  4808.3  651.63  4829.3  652.03  4857.7  648.17  4879.3  642.02
  4893.5  638.96  4928.7  636.88  5082.7  636.23    5148  636.87  5183.3  639.08
  5190.5  641.58  5197.4  642.09  5204.6  645.12  5218.8  646.83  5268.2  646.92
  5288.2  647.82  5317.8  649.16  5338.9  647.86  5358.8  647.85  5422.6  646.54
  5496.2  646.67  5563.7  647.31  5579.5  647.95  5593.6  649.93  5621.1  650.99
#Mann= 9 ,-1 , 0
  4574.5    .075       0  4801.8     .05       0  4928.7    .033       0
    5148     .05       0  5288.2    .075       0  5358.8     .05       0
  5422.6    .075       0  5496.2     .05       0  5563.7    .075       0
Bank Sta=4928.7,5148
XS Rating Curve= 0 ,0
Exp/Cntr=0.3,0.1

Type RM Length L Ch R = 1 ,16865   ,270,270,270
BEGIN DESCRIPTION:
Cade Branch 34.0
END DESCRIPTION:
XS GIS Cut Line= 3
      2355824.57      7049362.49      2356749.07      7048848.15
      2357289.43      7048496.59
#Sta/Elev= 30
  3929.3  652.72  4117.5   651.7  4163.2   650.6  4175.7  651.62  4326.4  651.33
  4609.5   652.4  4722.3  651.13  4857.7  651.18  4870.8  649.68  4874.4  649.76
  4884.2  647.69  4890.4  644.52  4896.1  644.71  4906.4  642.43  4912.1  642.31
  4918.5  639.97  4928.1  638.19  4975.5  636.35  5159.1  637.73  5166.1  639.48
  5174.2  642.78  5201.9   645.8  5225.6  643.37  5246.7  642.75  5311.7  643.67
  5382.5  644.95  5584.7  646.01  5593.9  645.46  5607.5  646.69  5631.9     647
#Mann= 7 ,-1 , 0
  3929.3    .075       0  4326.4      .1       0  4857.7    .075       0
  4870.8     .05       0  4928.1    .033       0  5159.1     .05       0
  5311.7    .075       0
Bank Sta=4928.1,5159.1
XS Rating Curve= 0 ,0
Exp/Cntr=0.3,0.1

Type RM Length L Ch R = 1 ,16595   ,68,68,68
BEGIN DESCRIPTION:
Cade Branch 33.0
END DESCRIPTION:
XS GIS Cut Line= 4
      2356812.03      7049761.75      2356828.02      7049735.69
      2356792.48      7049104.22      2357332.86      7048568.18
#Sta/Elev= 30
  4270.4  646.73    4301  646.28  4306.7  643.65  4336.7  637.05  4445.1  635.32
  5117.8  636.75  5124.9  637.65  5146.1  638.33  5160.2  640.25  5167.3  642.44
  5174.4  643.17  5181.5  645.14  5188.5  645.36  5202.7  644.85  5209.8  643.08
    5231  641.84  5252.2  642.05  5280.5  639.99  5301.7  641.08  5308.8  642.79
  5372.4  642.44  5462.7  643.57  5575.2  645.34  5591.6  645.05  5598.7  645.78
  5619.8  646.39    5634  646.33  5641.1  645.55  5669.4  647.02  5694.6  646.72
#Mann= 5 ,-1 , 0
  4270.4     .05       0  4336.7    .033       0  5117.8     .05       0
  5462.7    .075       0  5575.2     .05       0
Bank Sta=4336.7,5117.8
XS Rating Curve= 0 ,0
Exp/Cntr=0.3,0.1

Type RM Length L Ch R = 1 ,16527   ,57,57,57
BEGIN DESCRIPTION:
Cade Branch 32.6
END DESCRIPTION:
XS GIS Cut Line= 6
      2356729.05      7049935.95      2356928.45      7049682.17
      2356868.45      7049114.59       2356977.1      7049004.31
      2356981.97      7048941.07      2357137.35      7048790.06
#Sta/Elev= 30
  4322.3  646.52  4470.5  646.46  4475.5  644.71  4542.4  646.69  4634.7  644.61
  4661.9   645.7    4667  644.14  4703.8  645.77    4709  644.66  4757.1  645.52
  4798.4  646.31  4918.4  645.31  4953.1  643.01  4992.8  643.74  5006.9  642.28
  5105.9  641.49  5170.1  645.08  5184.8  643.97  5191.9  641.61  5241.4  641.66
  5260.7  639.79  5260.9  639.29  5264.7  639.79  5297.9  642.64  5305.1  641.81
  5312.1   642.7  5354.5  642.12  5471.7  643.93    5542  645.15  5653.7  646.49
#Mann= 7 ,-1 , 0
  4322.3     .05       0  4757.1     .12       0  4953.1     .05       0
  5260.7    .033       0  5264.7     .05       0  5471.7    .075       0
    5542     .05       0
Bank Sta=5260.7,5264.7
XS Rating Curve= 0 ,0
Exp/Cntr=0.3,0.1

Type RM Length L Ch R = 1 ,16470   ,293,293,293
BEGIN DESCRIPTION:
Cade Branch 32.4
END DESCRIPTION:
XS GIS Cut Line= 5
      2356936.12       7049700.5      2356927.46       7049515.9
      2356879.17      7049296.52      2356884.26      7049174.18
      2357369.72      7048735.31
#Sta/Elev= 30
  4390.5  646.22  4561.2  646.77    4653  645.55  4681.5  646.05  4686.6  645.16
  4704.2  645.97  4784.8  645.71  4913.8  644.66  4918.8  642.36  4928.9   642.4
  4935.8  640.18  4942.5  640.55    4950  639.07    5019  637.75  5019.2  637.25
    5023  637.75  5070.3  639.28  5122.7  638.87  5162.2  640.04  5190.6  639.44
    5219  641.23  5254.1  640.48  5332.6  642.11  5339.3  641.56  5424.5  643.97
  5438.7  645.31  5473.8  645.54    5488  644.71  5502.2  645.88  5576.8  646.18
#Mann= 5 ,-1 , 0
  4390.5     .05       0  4784.8     .12       0    5019     .07       0
    5023     .12       0  5122.7     .05       0
Bank Sta=5019,5023
XS Rating Curve= 0 ,0
Exp/Cntr=0.3,0.1

Type RM Length L Ch R = 1 ,16177   ,283,283,283
BEGIN DESCRIPTION:
Cade Branch 32.0
END DESCRIPTION:
XS GIS Cut Line= 4
      2356944.64      7049707.51      2356939.26      7049404.24
      2357183.04      7049353.75      2357374.85      7049180.43
#Sta/Elev= 30
    4605  643.06  4612.5   644.2  4639.2  646.85  4782.5  646.37  4792.5  645.39
  4832.5  644.85  4852.6  644.09  4902.6  639.81  4907.9  638.68  4910.7  638.68
  4918.3   636.6  4938.7  635.25  4977.5  634.75  4977.8  634.25  4981.3  634.25
  4981.5  634.75  5002.5  634.93  5049.2  635.38  5071.5  635.98  5081.7  636.55
  5099.4  638.61  5122.5  640.12  5185.4  641.32  5199.6  642.13  5222.6  642.47
  5234.7  642.26  5383.4  643.67  5397.6  643.38  5405.1  643.87  5415.8  643.89
#Mann= 5 ,-1 , 0
    4605     .05       0  4977.5    .033       0  4981.5     .05       0
  5002.5     .12       0  5222.6     .05       0
Bank Sta=4977.5,4981.5
XS Rating Curve= 0 ,0
Exp/Cntr=0.3,0.1

Type RM Length L Ch R = 1 ,15894   ,239,239,239
BEGIN DESCRIPTION:
Cade Branch 31.0
END DESCRIPTION:
XS GIS Cut Line= 3
      2356905.28      7049746.61      2357085.45      7049657.61
      2357544.74       7049367.3
#Sta/Elev= 30
  4769.4  643.94  4776.1  645.47  4792.9  642.57  4798.5  644.47    4807  642.31
  4815.4  640.83    4821  641.97  4829.3  640.14  4888.3  637.88  4901.6  636.41
  4918.5  634.85  4961.2  634.74  4961.4  634.24  4964.9  634.24  4965.2  634.74
  5057.4  635.01    5066  635.35  5087.2   637.7  5093.1   637.6  5108.4  638.22
  5116.5  639.06  5135.4   639.8    5152  640.29  5160.2  640.13  5166.1  640.62
  5211.2   640.9    5239  641.51  5442.5   642.9  5463.7  642.73  5513.7  643.57
#Mann= 5 ,-1 , 0
  4769.4     .05       0  4901.6     .12       0  4961.2     .07       0
  4965.2     .12       0  5135.4     .05       0
Bank Sta=4961.2,4965.2
XS Rating Curve= 0 ,0
Exp/Cntr=0.3,0.1

Type RM Length L Ch R = 1 ,15655   ,488,488,488
BEGIN DESCRIPTION:
Cade Branch 30.0
END DESCRIPTION:
XS GIS Cut Line= 3
      2356902.19       7049870.9      2357103.45      7049896.46
      2357479.02      7049659.99
#Sta/Elev= 30
    4752  641.53  4784.3  641.59  4789.3   640.8  4809.3  640.64  4829.4  641.25
  4849.6  642.44  4869.8  642.32  4879.8  640.05  4889.9  639.05  4977.8   636.2
  4997.2  634.52  5008.4   632.7  5020.5  631.86  5027.6  631.77  5027.8  631.27
  5031.3  631.27  5031.6  631.77  5079.6  632.31  5108.5  633.94  5129.7  634.44
    5145  636.04  5150.9  635.45  5160.2  636.08  5187.4  636.56  5258.7  638.86
  5312.1  639.51    5318  639.88  5369.8  640.31    5391  642.22  5398.7  642.16
#Mann= 5 ,-1 , 0
    4752     .05       0  4997.2    .075       0  5027.6     .07       0
  5031.6    .075       0  5258.7     .05       0
Bank Sta=5027.6,5031.6
XS Rating Curve= 0 ,0
Exp/Cntr=0.3,0.1

Type RM Length L Ch R = 1 ,15167   ,302,302,302
BEGIN DESCRIPTION:
Cade Branch 29.0
END DESCRIPTION:
XS GIS Cut Line= 3
      2356979.02        7050260.        2357379.        7050260.
      2357579.01        7050160.
#Sta/Elev= 30
  4595.5  641.36  4615.5  641.33  4625.5  640.86  4645.5  639.03  4665.5  638.42
  4725.5  638.06  4875.5  636.24  4895.5   635.2  4905.5  634.02  4925.5  630.92
  4935.5  629.87  4955.5  629.43  4975.5  629.72    4991  628.72  4991.2  628.22
  4994.7  628.22    4995  628.72  5000.3  628.75  5009.5  628.89  5017.8  629.58
  5026.2  629.63  5054.2  632.44  5070.9  633.01  5076.5  633.71  5098.9     635
  5121.3  635.93  5160.4  636.58  5182.8  637.31  5205.1   638.5  5219.1  638.95
#Mann= 4 ,-1 , 0
  4595.5     .05       0    4991    .033       0    4995     .05       0
  5000.3    .075       0
Bank Sta=4991,4995
XS Rating Curve= 0 ,0
Exp/Cntr=0.3,0.1

Type RM Length L Ch R = 1 ,14865   ,277,277,277
BEGIN DESCRIPTION:
Cade Branch 28.0
END DESCRIPTION:
XS GIS Cut Line= 3
      2357232.85      7050557.68      2357561.83        7050497.
      2357735.01      7050409.62
#Sta/Elev= 30
  4696.8  636.54  4709.9  636.27  4804.7  635.68  4855.6  634.97    4879  634.49
  4896.3  633.27  4937.1  631.76    4971  630.95    4990  629.88  4997.9  628.72
  5006.1  627.02  5006.4  626.52  5009.9  626.52  5010.1  627.02  5027.3   627.8
  5040.4  627.61  5050.6  627.92  5057.1  629.24  5062.7  629.49  5079.4  632.08
  5101.7  633.76    5124  634.82  5129.6  635.38  5151.9  636.84  5174.2  637.33
    5185  637.28  5190.9  637.68  5207.4  637.88  5218.8  638.65  5225.3  638.73
#Mann= 4 ,-1 , 0
  4696.8     .05       0    4971    .075       0  5006.1     .07       0
  5010.1    .075       0
Bank Sta=5006.1,5010.1
XS Rating Curve= 0 ,0
Exp/Cntr=0.3,0.1

Type RM Length L Ch R = 1 ,14588   ,48,48,48
BEGIN DESCRIPTION:
Cade Branch 27.4
END DESCRIPTION:
XS GIS Cut Line= 5
      2357213.67      7050575.26      2357418.09      7050631.16
      2357585.79      7050712.61      2357775.85      7050714.21
      2358069.77      7050640.73
#Sta/Elev= 30
  4504.8  636.38  4665.8  632.93  4752.5  632.08  4769.5  631.39  4775.1  632.28
  4792.1  630.78  4797.7  631.98  4814.7   629.9  4820.2  630.18  4833.7  629.27
  4842.8  629.78  4859.8  629.12  4865.3  629.53  4944.4  625.62  4944.6  625.12
  4948.1  625.12  4948.4  625.62  5056.4  627.59  5086.4  630.35  5092.3  631.77
  5131.9  633.33    5148  632.78    5168  633.28  5209.2  635.64  5230.5  635.27
  5313.9  636.68  5374.1  637.13  5385.1  638.12  5393.2  640.83  5396.2  640.83
#Mann= 5 ,-1 , 0
  4504.8     .05       0  4833.7    .075       0  4944.4     .07       0
  4948.4    .075       0  5313.9     .05       0
Bank Sta=4944.4,4948.4
XS Rating Curve= 0 ,0
Exp/Cntr=0.3,0.1

Type RM Length L Ch R = 1 ,14540   ,49,49,49
BEGIN DESCRIPTION:
Cade Branch 27.3
END DESCRIPTION:
XS GIS Cut Line= 5
      2357240.81       7050663.1       2357413.3       7050664.7
        2357581.      7050746.15      2357771.06      7050747.75
      2358063.08      7050674.75
#Sta/Elev= 30
  4505.8   637.6    4664   635.9  4701.6  636.38  4707.1   635.3  4724.1  636.33
  4729.7   635.5  4740.2  636.28  4752.3  635.77  4758.8  636.24  4784.7  635.94
  4791.8   634.6  4797.4  635.74  4806.9  634.86  4814.4  632.89    4820  634.58
    4837  632.67  4842.5  633.95  4859.5  633.05  4863.4  633.66  4962.7  632.14
  5065.1  631.81  5065.4  631.31  5069.1  631.81  5166.1  632.82  5190.8  635.41
  5207.3  634.32  5279.6  636.07  5341.3  636.81  5350.6  637.87  5355.8  639.54
#Mann= 5 ,-1 , 0
  4505.8     .05       0  4758.8    .075       0  5065.1     .07       0
  5069.1    .075       0  5279.6     .05       0
Bank Sta=5065.1,5069.1
XS Rating Curve= 0 ,0
Exp/Cntr=0.3,0.1

Type RM Length L Ch R = 1 ,14491   ,24,24,24
BEGIN DESCRIPTION:
Cade Branch 27.2
END DESCRIPTION:
XS GIS Cut Line= 4
      2357320.67      7050827.61      2357700.79      7050787.68
      2357745.51      7050795.67      2358072.89      7050698.25
#Sta/Elev= 30
    4589  636.57  4613.2  634.84  4674.2  633.37  4738.1   631.6  4778.4  633.87
  4788.4  632.58  4798.5  630.04  4804.5  629.55  4858.8  627.82    4889  624.69
  4895.6  624.63  4895.8  624.13  4899.3  624.13  4899.6  624.63  4919.1  626.38
  4929.2  626.56    5014  626.22    5062  629.87  5072.4  629.63  5103.7  631.08
  5145.5  631.62  5160.2  633.03  5198.6  634.54  5231.8  635.11  5249.8  634.69
    5270  635.54  5336.5   636.6  5343.7  637.93  5353.6  641.47  5358.2  641.47
#Mann= 5 ,-1 , 0
    4589      .1       0  4674.2    .075       0  4895.6     .07       0
  4899.6    .075       0    5270     .05       0
Bank Sta=4895.6,4899.6
XS Rating Curve= 0 ,0
Exp/Cntr=0.3,0.1

Type RM Length L Ch R = 1 ,14467   ,76,76,76
BEGIN DESCRIPTION:
Cade Branch 27.0
END DESCRIPTION:
XS GIS Cut Line= 4
      2357320.65      7050851.57      2357700.79      7050811.64
      2357745.51      7050819.62      2358072.96      7050722.19
#Sta/Elev= 30
  4596.6  636.18  4615.1  636.49  4625.1  635.09  4692.9  633.31  4765.9  631.03
  4806.1  632.21  4826.2  628.95  4866.4  627.43  4894.6  624.54  4894.8  624.04
  4898.6  624.54  4906.7  625.71  4949.3  625.79    4967   626.6  5028.7  625.63
  5048.8  627.37  5069.6  627.64  5075.2  629.43  5080.4  628.69  5090.5  629.96
  5113.6  630.31  5121.8  629.33  5132.2  629.52  5205.3  633.97    5277  634.84
  5340.9  636.02  5351.1  637.84  5356.3  637.92  5361.2  641.55  5365.9  641.55
#Mann= 5 ,-1 , 0
  4596.6      .1       0  4692.9    .075       0  4894.6     .07       0
  4898.6    .075       0    5277     .05       0
Bank Sta=4894.6,4898.6
XS Rating Curve= 0 ,0
Exp/Cntr=0.3,0.1

Type RM Length L Ch R = 1 ,14391   ,121,121,121
BEGIN DESCRIPTION:
Cade Branch 26.8
END DESCRIPTION:
XS GIS Cut Line= 3
      2357327.05      7051044.82      2357793.42      7050822.82
      2358075.05      7050748.04
#Sta/Elev= 30
  4609.4  637.12  4666.9  635.81  4703.9  632.36  4755.5  630.54  4794.7  631.47
  4800.2   630.1  4818.5  630.54  4845.7  628.57  4862.8  628.76  4899.5  624.05
  4923.9   624.4  4934.5     624  4934.7   623.5  4938.5     624  4958.9  624.13
  4981.9  625.01  4999.1  624.01  5004.6  625.44  5010.3   624.4  5072.7  624.73
  5118.2  628.47  5125.9  627.82  5131.7  629.11    5157  629.68  5173.1  628.76
  5232.1  633.05  5326.4  634.54  5392.8   635.7    5411  642.06  5417.3  647.44
#Mann= 7 ,-1 , 0
  4609.4      .1       0  4818.5    .075       0  4923.9      .1       0
  4934.5     .07       0  4938.5      .1       0  4958.9    .075       0
  5326.4     .05       0
Bank Sta=4934.5,4938.5
XS Rating Curve= 0 ,0
Exp/Cntr=0.3,0.1

Type RM Length L Ch R = 1 ,14270   ,67,67,67
BEGIN DESCRIPTION:
Cade Branch 26.6
END DESCRIPTION:
XS GIS Cut Line= 3
      2357346.19       7051121.5      2357914.81      7050856.36
      2358085.64      7050796.25
#Sta/Elev= 30
  4666.3   637.1  4669.7   637.1  4929.7  630.96  4940.8  630.47  4956.3  626.49
  4961.6  624.17  4961.9  623.67  4965.9  624.17  5022.8   625.1  5058.4  625.33
  5106.4  625.12  5111.9  626.14  5134.8  626.81  5152.2   625.7  5157.7  626.68
    5175   625.5  5180.5  627.17  5203.4   629.4  5210.1  630.88  5220.7  631.83
  5226.3   630.8  5232.1   632.5  5243.2  633.24  5331.6     633  5368.8   633.8
    5436  634.94  5444.8  638.18  5450.1  638.19  5467.8  647.91  5474.8  649.12
#Mann= 8 ,-1 , 0
  4666.3    .075       0  4669.7      .1       0  4929.7    .075       0
  4961.6     .07       0  4965.9    .075       0  5022.8      .1       0
  5058.4    .075       0  5368.8     .05       0
Bank Sta=4961.6,4965.9
XS Rating Curve= 0 ,0
Exp/Cntr=0.3,0.1

Type RM Length L Ch R = 1 ,14203   ,221,221,221
BEGIN DESCRIPTION:
Cade Branch 26.4
END DESCRIPTION:
XS GIS Cut Line= 3
      2357371.79      7051178.98      2357940.36      7050913.86
      2358112.85      7050853.16
#Sta/Elev= 30
  4642.5  637.12  4699.7  636.14  4768.3  633.69  4845.5  632.75  4875.7  632.27
  4933.8  630.67  4956.7  627.82  4962.2  625.79  4990.3  623.95  4990.7  623.45
  4994.3  623.45  4994.6  623.95  5036.6  624.83  5104.9  624.19  5145.1  624.49
  5150.7  625.51    5158  628.76    5168  630.77  5202.1  632.74  5242.1  631.59
  5316.1  632.38  5342.6  633.89  5374.4  633.74  5383.3  635.34  5388.6  635.18
  5414.3  648.31  5419.6  648.23  5427.4  649.06  5445.2  645.67  5452.7  645.59
#Mann= 6 ,-1 , 0
  4642.5    .075       0  4845.5      .1       0  4875.7    .075       0
  4990.3     .07       0  4994.6    .075       0  5316.1     .05       0
Bank Sta=4990.3,4994.6
XS Rating Curve= 0 ,0
Exp/Cntr=0.3,0.1

Type RM Length L Ch R = 1 ,13982   ,107,107,107
BEGIN DESCRIPTION:
Cade Branch 26.2
END DESCRIPTION:
XS GIS Cut Line= 3
      2357470.76      7051246.08      2358039.39      7050980.94
      2358211.92      7050920.23
#Sta/Elev= 30
  4555.5  634.51  4693.4  630.79  4786.9  628.25  4798.3  629.46  4815.6  627.69
  4821.1  629.99  4838.5  626.74    4844  627.92  4861.3  626.33  4866.8  627.78
  4913.2  625.24    4941  625.02  4992.8  622.31  4993.1  621.81  4997.1  622.31
  5026.9  624.94  5032.4  626.73  5049.8  625.66  5055.3  627.69  5078.1  626.02
    5101   626.8  5106.5  628.48  5118.7  627.83  5129.4  628.82  5146.7  627.91
  5152.3  629.57  5169.6  629.17  5175.1  630.21  5230.6   630.5  5365.8  636.26
#Mann= 7 ,-1 , 0
  4555.5    .075       0  4693.4      .1       0  4786.9     .05       0
  4913.2    .075       0  4992.8     .07       0  4997.1    .075       0
  5118.7     .05       0
Bank Sta=4992.8,4997.1
XS Rating Curve= 0 ,0
Exp/Cntr=0.3,0.1

Type RM Length L Ch R = 1 ,13875   ,416,416,416
BEGIN DESCRIPTION:
Cade Branch 26.0
END DESCRIPTION:
XS GIS Cut Line= 3
      2357614.57      7051292.37      2358183.13      7051027.25
      2358354.78      7050966.86
#Sta/Elev= 30
  4663.5  633.15  4677.8  633.63  4690.5  634.27  4734.6  632.68  4774.4  633.37
  4779.9  632.32  4797.3  632.98  4802.8  631.24  4820.1  632.24  4825.7   631.1
  4865.9  631.07  4871.4  629.72  4888.7  630.82  4894.2  629.26  4911.1  630.47
  4922.6  629.42  4977.3  629.58  5008.6  626.53  5014.1  621.95  5034.8  621.78
  5035.2  621.28  5039.1  621.78  5098.7  623.92  5128.4  627.27  5294.7  627.94
  5318.3  629.87    5331  631.97  5387.6   633.7  5392.9  635.23  5472.8  636.77
#Mann= 4 ,-1 , 0
  4663.5    .075       0  4677.8     .05       0  5034.8     .05       0
  5039.1     .05       0
Bank Sta=5034.8,5039.1
XS Rating Curve= 0 ,0
Exp/Cntr=0.3,0.1

Type RM Length L Ch R = 1 ,13459   ,459,459,459
BEGIN DESCRIPTION:
Cade Branch 25.0
END DESCRIPTION:
XS GIS Cut Line= 3
      2357806.16       7051351.5      2358243.82      7051163.01
      2358483.43      7051113.49
#Sta/Elev= 30
  4486.5  634.63    4499  634.43  4504.4  632.76    4528     633  4533.4  631.37
  4551.5  631.79  4556.9  630.53  4627.5  629.98    4633  629.29  4685.6  628.19
  4703.5  628.97    4709  627.99  4727.1  628.73  4732.5  627.83  4750.6  628.87
    4756  627.92  4779.6  628.45    4785  627.07  4795.1  626.39  4855.6  621.71
  4937.1  622.56  4986.5  620.18  4986.9  619.68    4991  620.18  4998.2   622.8
  5003.3   622.9  5009.2  626.98  5048.6  628.52  5103.8  631.06  5207.7  633.23
#Mann= 5 ,-1 , 0
  4486.5     .05       0  4795.1     .12       0  4986.5     .07       0
    4991     .12       0  5048.6     .05       0
Bank Sta=4986.5,4991
XS Rating Curve= 0 ,0
Exp/Cntr=0.3,0.1

Type RM Length L Ch R = 1 ,13000   ,180,180,180
BEGIN DESCRIPTION:
Cade Branch 24.0
END DESCRIPTION:
XS GIS Cut Line= 3
      2358063.35       7051787.5      2358411.53      7051362.66
      2358526.46      7051084.89
#Sta/Elev= 30
  4472.1  637.09  4481.8  636.71  4488.6   634.1  4517.3   629.5  4531.6  629.13
  4609.9  627.78  4688.1  627.59  4694.6  628.12  4772.8  627.81  4879.7   629.3
  4894.1  628.57  4908.4  625.12  4914.9  622.35  4921.4  620.76  4951.4  619.81
  4978.8  619.36    4986  618.24  4993.1  618.58  4997.3  618.02  4997.8  617.52
  5001.9  618.02  5007.5  619.48  5076.6  619.91  5159.1  619.33  5175.8  622.12
  5185.7  624.87  5197.4  627.37  5219.1  629.67  5265.5  632.16    5322  633.68
#Mann= 5 ,-1 , 0
  4472.1     .05       0  4951.4     .12       0  4997.3     .07       0
  5001.9     .12       0  5185.7     .05       0
Bank Sta=4997.3,5001.9
XS Rating Curve= 0 ,0
Exp/Cntr=0.3,0.1

Type RM Length L Ch R = 1 ,12820   ,98,98,98
BEGIN DESCRIPTION:
Cade Branch 23.2
END DESCRIPTION:
XS GIS Cut Line= 3
      2358219.22       7051778.9       2358491.9      7051609.86
      2358654.19      7051175.52
#Sta/Elev= 30
  4464.6  629.68  4513.6   629.4  4565.6  629.97  4644.8   629.3  4821.3  630.11
  4838.7  629.34  4846.3  627.92  4851.6  627.59  4870.7  619.95  4876.6   618.7
  4897.9  618.01  4943.1  617.64  4943.6  617.14  4947.3  617.14  4947.7  617.64
  4962.1  618.39  4992.4  617.79  5017.4  618.45  5022.7  618.14  5030.8  619.96
  5041.5  623.13  5047.7  623.96  5116.2  624.39  5133.3  624.89  5143.6  626.03
  5188.5  627.36  5218.8  627.63  5224.1  628.51  5233.6  629.22  5249.1  629.03
#Mann= 5 ,-1 , 0
  4464.6     .05       0  4897.9     .12       0  4943.1     .07       0
  4947.7     .12       0  5143.6     .05       0
Bank Sta=4943.1,4947.7
XS Rating Curve= 0 ,0
Exp/Cntr=0.3,0.1

Type RM Length L Ch R = 1 ,12722   ,36,36,36
BEGIN DESCRIPTION:
Cade Branch 23.1
END DESCRIPTION:
XS GIS Cut Line= 3
      2358274.61      7051815.99      2358547.29      7051646.96
       2358710.2      7051210.91
#Sta/Elev= 30
  4391.7   629.7  4675.8  630.66  4733.8  628.86  4759.3  629.18  4789.1  625.82
  4805.3  626.63  4819.4  625.62  4880.1   626.2  4904.9  625.48  4954.8  626.46
  4960.2  625.92  4965.5  627.09  4976.1  626.76  4985.2  621.52  4995.2  617.77
  4995.6  617.27  4999.8  617.77  5008.2  617.83  5015.5  619.62  5020.8  622.71
  5029.5  624.48  5061.5  624.78  5070.7  625.39  5076.1  627.49  5082.1  626.53
  5131.3  626.38  5146.9  627.85  5156.3  629.64  5161.6  631.95    5178  633.04
#Mann= 5 ,-1 , 0
  4391.7     .05       0  4759.3     .12       0  4995.2     .07       0
  4999.8     .12       0  5082.1     .05       0
Bank Sta=4995.2,4999.8
XS Rating Curve= 0 ,0
Exp/Cntr=0.3,0.1

Type RM Length L Ch R = 1 ,12686   ,478,478,478
BEGIN DESCRIPTION:
Cade Branch 23.0
END DESCRIPTION:
XS GIS Cut Line= 3
      2358308.17      7051843.12      2358612.18      7051618.54
      2358721.75      7051226.84
#Sta/Elev= 30
  4399.9   629.3  4495.9  630.52    4711  630.08  4761.1  627.71  4772.8  625.47
  4777.9  625.47  4783.1  621.35  4788.3  618.38  4792.5  618.03  4805.2  617.51
  4805.7  617.01  4809.4  617.01  4809.8  617.51  4861.7  618.25  4963.3  617.84
  4969.3  619.46  4974.5  617.67  5003.5   617.7  5008.7  618.81  5015.2  619.16
  5025.6  622.64    5048  623.45  5079.3  626.62  5087.9   627.1  5116.3  626.41
  5121.5  627.19  5139.8  627.73  5155.6  630.06  5160.8  631.44  5184.6  632.82
#Mann= 5 ,-1 , 0
  4399.9     .05       0  4792.5     .12       0  4805.2     .07       0
  4809.8     .12       0  5079.3     .05       0
Bank Sta=4805.2,4809.8
XS Rating Curve= 0 ,0
Exp/Cntr=0.3,0.1

Type RM Length L Ch R = 1 ,12208   ,491,491,491
BEGIN DESCRIPTION:
Cade Branch 22.0
END DESCRIPTION:
XS GIS Cut Line= 2
      2358330.04      7051895.17      2358967.28      7051774.84
#Sta/Elev= 30
    4390  629.92  4419.5  629.99    4450  630.66  4480.5   630.4  4497.3  629.54
  4521.2  629.36  4664.6  630.22  4769.4  629.49  4806.2  628.09  4816.4  626.54
  4821.8  624.02  4826.8  624.57  4833.4  621.11  4836.7  619.38  4846.9  618.92
  4857.1  619.33  4874.1  617.07  4879.2  618.24  4897.8  619.17  4931.6  618.04
  4958.8  615.55    4984  613.79  4987.1  612.09  4987.5  611.59  4991.2  611.59
  4991.7  612.09  5009.7  615.99  5019.9  620.86  5023.4  621.83  5038.5  625.79
#Mann= 5 ,-1 , 0
    4390     .05       0  4833.4     .12       0  4987.1     .07       0
  4991.7     .12       0  5023.4     .05       0
Bank Sta=4987.1,4991.7
XS Rating Curve= 0 ,0
Exp/Cntr=0.3,0.1

Type RM Length L Ch R = 1 ,11717   ,296,296,296
BEGIN DESCRIPTION:
Cade Branch 21.0
END DESCRIPTION:
XS GIS Cut Line= 3
       2358535.5       7052412.8      2358727.21      7052221.09
      2359027.29      7051893.73
#Sta/Elev= 30
  4643.4  630.48  4690.3  628.13  4768.1   627.8  4810.5  623.74  4874.1  622.61
  4881.2  621.36  4902.4  621.98  4909.5  618.37  4912.2  619.36  4918.6  619.36
  4923.7  613.48  4930.5   616.8  4937.9  612.38  4944.6  612.94    4952  610.86
  4958.8  611.94  4963.9  610.36  4964.4  609.86  4968.6  610.36    4973   611.9
  4989.7  611.84  5015.5  611.39  5037.1  612.83  5065.2  612.91  5100.6  616.29
  5240.3  618.16  5320.2  618.39  5339.4  622.29  5355.3  624.06  5358.6  623.48
#Mann= 6 ,-1 , 0
  4643.4     .05       0  4963.9     .07       0  4968.6     .05       0
  4989.7     .12       0  5240.3     .05       0  5339.4     .12       0
Bank Sta=4963.9,4968.6
XS Rating Curve= 0 ,0
Exp/Cntr=0.3,0.1

Type RM Length L Ch R = 1 ,11421   ,213,213,213
BEGIN DESCRIPTION:
Cade Branch 20.2
END DESCRIPTION:
XS GIS Cut Line= 4
      2359121.61      7052445.68      2359110.65      7052237.52
      2359035.62      7052041.79      2359017.54      7051930.82
#Sta/Elev= 30
  4707.9  617.91  4813.7  616.33  4833.8  614.79  4843.8  615.38  4850.7  614.78
  4855.7  615.49  4873.8  614.42  4903.8  611.33  4932.3  610.07  4937.7  610.89
  4956.5  611.15  4962.4  607.76  4967.7  612.09  4987.1  610.02  4992.4  611.58
  5022.4  609.77  5029.1  605.63  5029.6  605.13  5033.8  605.63  5047.1  609.34
  5063.6  612.24    5085  614.88  5109.9  616.01  5134.4   615.6  5139.5  617.26
  5168.3  616.48  5195.9  618.45    5201  617.81  5208.8  618.26  5238.4  620.94
#Mann= 5 ,-1 , 0
  4707.9     .05       0  4903.8     .12       0  5029.1     .07       0
  5033.8     .12       0  5109.9     .05       0
Bank Sta=5029.1,5033.8
XS Rating Curve= 0 ,0
Exp/Cntr=0.3,0.1

Type RM Length L Ch R = 1 ,11208   ,261,261,261
BEGIN DESCRIPTION:
Cade Branch 20.0
END DESCRIPTION:
XS GIS Cut Line= 3
      2359244.85      7052429.23       2359233.9      7052221.09
      2359108.42      7051893.75
#Sta/Elev= 30
  4830.5  614.74  4845.8  616.74  4850.8   614.3  4889.8  618.22  4899.8  618.49
  4909.8  618.28  4919.7  617.07  4939.9  615.23  4949.9  613.57  4959.9  613.05
  4969.9  610.45  4979.9  606.41  4987.6  604.56  4988.1  604.06  4992.4  604.56
    5010  607.66    5030  608.65  5038.9  610.27  5066.7  609.94  5115.1  610.87
  5160.2  613.94  5176.2  614.44  5181.5  615.47    5190   615.9  5206.2  615.44
  5211.5  616.83  5230.9  616.39  5236.2  617.22  5297.1  619.71  5389.5  620.18
#Mann= 5 ,-1 , 0
  4830.5     .05       0  4919.7     .12       0  4987.6     .07       0
  4992.4     .12       0  5160.2     .05       0
Bank Sta=4987.6,4992.4
XS Rating Curve= 0 ,0
Exp/Cntr=0.3,0.1

Type RM Length L Ch R = 1 ,10947   ,493,493,493
BEGIN DESCRIPTION:
Cade Branch 19.0
END DESCRIPTION:
XS GIS Cut Line= 3
      2359275.01      7052544.25       2359431.1      7052399.12
      2359803.59      7052108.79
#Sta/Elev= 30
  4798.2  619.92  4804.3  619.92  4811.1  616.12    4818  614.61  4825.3  614.29
  4839.5  617.11  4846.3  616.72  4860.5  613.44  4874.6  606.43    4882  605.16
  4895.1  605.96  4957.5  606.03  4978.8  604.69  4979.3  604.19  4983.6  604.69
  4994.8  605.21  5002.2  607.25  5037.3  607.29  5059.4  609.55  5101.6  616.01
  5140.8  615.14  5152.6  614.97  5180.3  614.34  5201.1  612.68    5230  614.25
  5300.6  614.32  5337.7  615.45    5351  617.28  5422.7  620.89  5483.6  622.34
#Mann= 7 ,-1 , 0
  4798.2     .05       0  4895.1     .12       0  4957.5     .05       0
  4978.8    .033       0  4983.6     .05       0  5140.8    .075       0
  5152.6     .05       0
Bank Sta=4978.8,4983.6
XS Rating Curve= 0 ,0
Exp/Cntr=0.3,0.1

Type RM Length L Ch R = 1 ,10454   ,378,378,378
BEGIN DESCRIPTION:
Cade Branch 18.5
END DESCRIPTION:
XS GIS Cut Line= 3
      2359306.36      7052941.39      2359656.33       7052791.4
      2360055.19      7052591.97
#Sta/Elev= 30
  4616.4   616.8  4739.3  613.27  4757.4  614.93  4762.8  614.59  4771.6  612.11
    4781  611.92  4793.3  614.17  4804.2  613.38    4810  610.61  4833.6  611.67
  4872.7  608.49  4886.1  607.98  4891.6  606.42  4915.2  604.58  4933.3  604.22
  4938.7  605.08  4956.5  602.62    4972  602.86  4983.2  601.64    4984  601.14
  4988.5  601.64  4995.9  603.81    5031  603.66  5075.7   608.6  5178.1  612.38
  5180.8  612.42  5215.4  613.08  5292.9  611.85  5328.9  612.45  5443.1  615.85
#Mann= 9 ,-1 , 0
  4616.4     .05       0  4872.7     .12       0    4972     .05       0
  4983.2    .033       0  4988.5     .05       0  5178.1    .075       0
  5180.8      .1       0  5292.9    .075       0  5328.9      .1       0
Bank Sta=4983.2,4988.5
XS Rating Curve= 0 ,0
Exp/Cntr=0.3,0.1

Type RM Length L Ch R = 1 ,10076   ,384,384,384
BEGIN DESCRIPTION:
Cade Branch 18.0
END DESCRIPTION:
XS GIS Cut Line= 3
      2359379.04      7052960.58      2359863.84      7053122.17
      2360284.85      7053144.05
#Sta/Elev= 30
  4525.7   615.3  4603.8  613.57  4667.1  609.39  4683.8  613.21  4698.7  613.04
    4725  607.38  4730.3  608.02  4736.5  604.56  4756.7  602.05  4825.2  602.74
  4851.5  604.66  4856.8  603.38    4863  605.05  4894.6  605.76  4914.8  605.31
  4920.1  603.63  4926.2  605.41  4936.8  606.09  4986.8   600.4  4987.6   599.9
  4992.2   600.4    5000   601.9  5016.8  601.57  5094.1     604    5142  611.07
  5185.4  611.11  5222.1  609.22  5280.6  616.31  5342.3  618.38  5458.3  618.11
#Mann= 6 ,-1 , 0
  4525.7     .05       0    4725     .12       0  4986.8     .07       0
  4992.2     .12       0  5016.8     .05       0  5185.4    .075       0
Bank Sta=4986.8,4992.2
XS Rating Curve= 0 ,0
Exp/Cntr=0.3,0.1

Type RM Length L Ch R = 1 ,9692    ,88,88,88
BEGIN DESCRIPTION:
Cade Branch 17.0
END DESCRIPTION:
XS GIS Cut Line= 4
      2359373.56      7053021.93      2359617.34      7053093.14
      2359850.14      7053556.01       2360072.8      7053660.65
#Sta/Elev= 30
  4352.5  614.85  4396.9  614.42  4430.3  612.87  4435.5   611.3  4462.3  611.81
  4514.4  609.01  4535.3  611.05  4541.1  613.22  4556.1  612.97  4574.6  606.34
  4579.8  608.06  4587.4  604.14  4599.8     602  4620.5  603.87  4626.1  602.96
  4642.8  605.23  4651.1  604.44  4687.5  605.72  4804.7  604.68  4991.7  599.82
  4992.5  599.32  4997.1  599.82    5039  603.11  5126.7  604.75  5165.6  606.99
  5188.4  607.18  5211.2  602.18  5239.6  608.37  5285.2  611.03  5370.6  613.23
#Mann= 5 ,-1 , 0
  4352.5     .05       0  4599.8     .12       0  4651.1     .05       0
  4991.7     .05       0  4997.1     .05       0
Bank Sta=4991.7,4997.1
XS Rating Curve= 0 ,0
Exp/Cntr=0.3,0.1

Type RM Length L Ch R = 1 ,9604    ,160,160,160
BEGIN DESCRIPTION:
Cade Branch 16.5
END DESCRIPTION:
XS GIS Cut Line= 4
      2359296.91      7053101.36      2359540.65      7053172.57
      2359767.98      7053568.61      2359828.04       7053649.1
#Sta/Elev= 30
  4358.5  618.22    4569  609.44  4719.3   608.1  4740.9  606.35  4880.4  604.93
  4939.3  602.47  4955.1  602.44  4960.9  604.38  4976.7   602.2  4982.5   603.7
  4998.3  599.57  5017.1  599.45  5017.9  598.95  5022.5  599.45  5035.7  601.12
  5041.4  604.25  5047.6  605.25  5057.2  604.11    5063  607.54  5078.1  604.44
  5084.3  607.93  5092.7   606.5  5098.9  610.65  5107.3   608.9  5113.5  610.88
  5128.1  608.25  5134.4  610.88  5142.7  609.47    5149  610.97  5169.5  611.28
#Mann= 3 ,-1 , 0
  4358.5     .05       0  5017.1     .05       0  5022.5     .05       0
Bank Sta=5017.1,5022.5
XS Rating Curve= 0 ,0
Exp/Cntr=0.3,0.1

Type RM Length L Ch R = 1 ,9444    ,109,109,109
BEGIN DESCRIPTION:
Cade Branch 16.2
END DESCRIPTION:
XS GIS Cut Line= 3
      2359135.26      7053554.91      2359661.16      7053650.77
      2359832.49      7053651.65
#Sta/Elev= 30
    4349  620.83  4383.3  619.09  4407.4  618.99  4454.4  618.84  4470.6  618.02
  4505.3  617.27  4525.6  615.18  4545.9   615.3  4586.6  613.26  4637.4  612.57
  4678.1  610.05  4698.4  610.03  4749.2  608.64  4795.3  609.13  4808.4   608.4
  4883.6  607.59  4911.4  603.92  4931.4  603.14  4961.4  602.87  4981.4  603.37
  4991.4  602.44  4998.7  598.71  4999.5  598.21  5003.3  598.21  5004.1  598.71
  5011.4  600.46  5021.4   604.1  5031.4  606.67  5041.4  610.57  5054.9  611.28
#Mann= 6 ,-1 , 0
    4349    .075       0  4407.4     .05       0  4470.6    .075       0
  4808.4     .05       0  4998.7     .05       0  5004.1     .05       0
Bank Sta=4998.7,5004.1
XS Rating Curve= 0 ,0
Exp/Cntr=0.3,0.1

Type RM Length L Ch R = 1 ,9335    ,121,121,121
BEGIN DESCRIPTION:
Cade Branch 16.0
END DESCRIPTION:
XS GIS Cut Line= 3
      2359050.37      7054068.19      2359789.89      7053723.08
      2359849.24      7053696.76
#Sta/Elev= 30
  4220.2     622  4231.5  620.81  4248.8  619.97  4254.3  620.51  4345.8  616.31
    4397  615.23  4437.2  612.95  4442.7  613.16  4460.1  612.22  4516.8  610.93
  4585.4     608  4676.8  606.06  4847.9  605.14  4939.3   604.1    4947  603.47
  4962.2  603.71  4969.1  602.49  4979.5  599.04    4985  599.19  4988.5  598.65
  4989.2  598.15  4993.1  598.15  4993.9  598.65  5002.2  602.74  5007.9  603.87
  5059.4  604.38  5082.7  605.95    5090  608.81  5098.4  610.93  5101.2  610.93
#Mann= 3 ,-1 , 0
  4220.2     .05       0  4988.5     .05       0  4993.9     .05       0
Bank Sta=4988.5,4993.9
XS Rating Curve= 0 ,0
Exp/Cntr=0.3,0.1

Type RM Length L Ch R = 1 ,9214    ,167,167,167
BEGIN DESCRIPTION:
Cade Branch 15.6
END DESCRIPTION:
XS GIS Cut Line= 4
       2358984.7       7054231.4      2359411.93      7054078.04
      2359820.01       7053828.8      2359902.21      7053790.44
#Sta/Elev= 30
  4113.6  624.68    4128  624.44  4133.3  625.68  4158.7  623.02  4164.1  623.22
  4171.3  621.29  4189.5  618.68  4194.8  619.34  4220.2  616.88  4225.5   617.4
  4245.6  616.04    4251  616.38  4276.4  614.99  4281.7  615.36  4312.4  614.38
  4424.7  610.07  4491.5  609.26  4563.3   606.7    4651  605.45  4745.9  603.16
  4962.7  603.41  5006.4  597.64  5007.1  597.14  5011.8  597.64  5030.4  602.87
  5066.7  603.85  5103.6  606.03    5121  610.46  5126.5  610.89  5136.4  610.23
#Mann= 3 ,-1 , 0
  4113.6     .05       0  5006.4     .05       0  5011.8     .05       0
Bank Sta=5006.4,5011.8
XS Rating Curve= 0 ,0
Exp/Cntr=0.3,0.1

Type RM Length L Ch R = 1 ,9047    ,118,118,118
BEGIN DESCRIPTION:
Cade Branch 15.0
END DESCRIPTION:
XS GIS Cut Line= 3
      2358998.36      7054320.15      2359773.45      7054029.83
      2359967.96      7053949.29
#Sta/Elev= 30
  4076.5  626.26  4117.1  625.94  4122.5  625.26  4141.3  621.64  4147.4  617.96
  4162.6  615.41  4202.6  613.76  4207.9  614.06  4263.1  612.64  4343.3  608.97
  4434.1  607.36  4489.3  604.97  4494.6  605.31  4574.8   603.2  4660.3  601.97
  4831.2  601.19  4969.4  601.92  4975.1  599.98  4983.2   596.2    4984   595.7
  4987.9   595.7  4988.6   596.2  4993.3  597.42  4998.7  599.76  5007.6  602.07
  5046.5  605.12  5094.2  607.32  5099.7  608.74  5105.1  608.97  5114.7  610.63
#Mann= 3 ,-1 , 0
  4076.5     .05       0  4983.2    .033       0  4988.6     .05       0
Bank Sta=4983.2,4988.6
XS Rating Curve= 0 ,0
Exp/Cntr=0.3,0.1

Type RM Length L Ch R = 1 ,8929    ,458,458,458
BEGIN DESCRIPTION:
Cade Branch 14.2
END DESCRIPTION:
XS GIS Cut Line= 3
      2359042.14      7054403.97      2359735.11       7054160.2
      2360015.63      7054056.71
#Sta/Elev= 30
  4111.5  625.64  4129.4  625.37  4150.6  619.27  4161.2   617.6  4167.6  613.73
  4198.5  611.32  4203.8  611.65    4246  610.05  4322.4  608.38    4410  605.43
    4458  603.14  4528.6  600.98  4616.2   599.5  4659.4  599.47  4678.1  598.83
  4714.4  600.11  4845.5  601.21  4913.9  600.68  4988.8  600.89  4999.5  599.26
  5007.8   595.3  5008.6   594.8  5012.5   594.8  5013.2   595.3  5020.8  596.25
  5030.3  599.63  5042.1  601.95  5091.2  605.89  5127.4  606.89  5145.1  609.06
#Mann= 3 ,-1 , 0
  4111.5     .05       0  5007.8     .05       0  5013.2     .05       0
Bank Sta=5007.8,5013.2
XS Rating Curve= 0 ,0
Exp/Cntr=0.3,0.1

Type RM Length L Ch R = 1 ,8471    ,715,715,715
BEGIN DESCRIPTION:
Cade Branch 14.0
END DESCRIPTION:
XS GIS Cut Line= 3
      2359085.98      7054531.05      2359784.41      7054331.11
      2360077.44      7054160.22
#Sta/Elev= 30
  4487.9  617.15  4508.3  615.09  4513.5  616.65  4532.6  612.06    4542  611.37
  4678.3  609.62  4782.3  603.55  4944.7  597.02  4949.9  597.78  4969.5  596.33
  4983.7  593.56  4987.6  591.32  4988.4  590.82  4993.1  591.32  5011.1  592.66
  5022.6  596.36  5031.9   596.9  5051.2  595.72  5056.4   597.9  5090.2  594.57
  5095.4  596.42    5124  594.07  5129.2  595.77  5162.9  593.74  5214.2  600.99
  5321.9  601.98  5429.4  604.88  5503.9  605.29  5519.6  604.49  5553.6  610.06
#Mann= 3 ,-1 , 0
  4487.9     .05       0  4987.6     .05       0  4993.1     .05       0
Bank Sta=4987.6,4993.1
XS Rating Curve= 0 ,0
Exp/Cntr=0.3,0.1

Type RM Length L Ch R = 1 ,7756    ,542,542,542
BEGIN DESCRIPTION:
Cade Branch 13.5
END DESCRIPTION:
XS GIS Cut Line= 3
      2359157.23      7054618.69      2359828.23      7054657.03
      2360249.34      7054454.68
#Sta/Elev= 30
  4142.9  609.57  4294.9  607.47  4515.3  602.22  4602.3  598.67  4615.4  599.35
  4675.5  598.34  4775.1     595  4780.1  595.44  4817.3  593.83  4862.9  590.54
  4863.9  590.04  4868.7  590.54  4871.4  591.33  4888.5   591.5  4993.4  590.74
  5007.2  592.44  5037.7  597.92  5069.6  600.56  5075.1  600.14  5092.2  601.43
  5097.8  601.01  5137.5  603.33    5143  602.76  5165.7  604.29  5193.9  603.96
  5248.5   605.2  5261.8  606.61  5270.7   609.5  5278.9  609.79  5282.2  609.04
#Mann= 3 ,-1 , 0
  4142.9     .05       0  4862.9    .033       0  4868.7     .05       0
Bank Sta=4862.9,4868.7
XS Rating Curve= 0 ,0
Exp/Cntr=0.3,0.1

Type RM Length L Ch R = 1 ,7214    ,647,647,647
BEGIN DESCRIPTION:
Cade Branch 13.0
END DESCRIPTION:
XS GIS Cut Line= 4
      2359212.01      7054783.02      2359771.63      7054825.53
        2360079.        7054960.      2360278.97        7054960.
#Sta/Elev= 30
  4102.8  607.22  4126.9  605.31  4200.1  605.26  4258.1  603.67  4520.5  600.18
  4571.1   598.6  4611.2  598.36  4656.7  596.27    4664  596.51  4704.8  595.02
  4740.3  593.02  4758.2  590.33  4781.2   588.3  4810.5  588.48  4830.9  587.86
  4831.8  587.36  4835.8  587.36  4836.7  587.86  4909.5  589.32  4923.1  589.35
    4945  588.23    5002  588.36  5009.5  590.09  5029.5  593.18  5039.5  595.92
  5049.5  597.64  5059.5  599.13  5070.1  599.51  5119.5  601.52  5199.5  603.55
#Mann= 4 ,-1 , 0
  4102.8     .05       0  4830.9    .033       0  4836.7     .05       0
  5070.1     .12       0
Bank Sta=4830.9,4836.7
XS Rating Curve= 0 ,0
Exp/Cntr=0.3,0.1

Type RM Length L Ch R = 1 ,6567    ,660,660,660
BEGIN DESCRIPTION:
Cade Branch 12.5
END DESCRIPTION:
XS GIS Cut Line= 4
      2359222.96      7055078.82       2359663.9       7055119.9
      2359925.47      7055403.26      2360165.96      7055358.53
#Sta/Elev= 30
  4269.9  603.96    4286  602.65  4338.9  601.75  4366.4  600.32  4436.7  594.86
    4443  595.95    4448  595.11  4496.9  595.19  4567.2  591.77  4587.3  591.83
  4617.4  593.82  4627.5  591.71  4647.6  593.76  4656.3  592.88  4667.7   589.7
  4712.8  590.77  4780.4  585.63  4808.2  586.24  4829.7  585.28  4992.4  585.39
  5020.8   584.9    5032  583.42    5033  582.92  5037.9  583.42  5063.3  591.21
  5070.1  592.34  5112.1  592.22    5224  595.92  5274.9  599.43    5343   600.1
#Mann= 3 ,-1 , 0
  4269.9     .05       0    5032    .033       0  5037.9     .05       0
Bank Sta=5032,5037.9
XS Rating Curve= 0 ,0
Exp/Cntr=0.3,0.1

Type RM Length L Ch R = 1 ,5907    ,444,444,444
BEGIN DESCRIPTION:
Cade Branch 12.0
END DESCRIPTION:
XS GIS Cut Line= 3
      2359105.19      7055533.46      2359778.93      7055462.25
       2360155.4       7055388.6
#Sta/Elev= 30
    4624  595.58  4665.8  594.56  4703.9  593.78  4708.9  594.77  4728.4  593.53
  4778.7  593.21  4796.7  591.99  4801.7  592.73  4828.9  591.77  4849.1  592.06
  4879.2  590.27  4894.6  586.01  4899.6  586.34  4909.4  585.04  4929.5  584.19
  4969.7  583.47  4979.8  581.19  4984.4  579.41  4985.4  578.91  4990.3  579.41
  4992.4  583.49  4999.9  581.83  5009.9   582.2  5030.1  586.41  5040.1  586.93
    5434  590.39  5556.3  594.43  5607.3  596.84  5637.8   599.2  5685.1  599.69
#Mann= 4 ,-1 , 0
    4624    .075       0  4665.8     .05       0  4984.4    .033       0
  4990.3     .05       0
Bank Sta=4984.4,4990.3
XS Rating Curve= 0 ,0
Exp/Cntr=0.3,0.1
