HEC-RAS study Elizabeth Creek.prj: Elizabeth Creek Base Level Engineering

--- Elizabeth Creek.g01 (geometry) --- (continued)

Type RM Length L Ch R = 1,89607,443,443,443
BEGIN DESCRIPTION:
Elizabeth Creek 101.0
END DESCRIPTION:
XS GIS Cut Line= 3
      2301018.58      7067169.83      2299392.17      7066243.15
      2298875.29      7066098.17
#Sta/Elev= 30
  3130.8  813.84  3291.4  811.30  3342.9  813.06  3407.7  809.77  3504.3  808.05
  3811.1  804.97  4574.7  800.91  4836.0  797.04  4881.6  797.40  4891.2  799.43
  4897.5  798.02  4903.2  799.67  4913.3  797.63  4983.9  795.69  4994.0  791.50
  4996.0  791.00  5011.4  791.50  5016.4  791.87  5026.7  797.08  5032.4  797.81
  5099.4  797.36  5105.8  796.90  5111.0  793.63  5134.2  792.78  5151.4  792.44
  5192.9  799.56  5234.5  802.73  5265.6  807.08  5392.4  810.96  5539.5  813.85
#Mann=6,-1,0
  3130.8    0.05       0  4836.0    0.12       0  4994.0    0.07       0
  5011.4    0.12       0  5134.2    0.05       0  5392.4    0.12       0
Bank Sta=4994,5011.4
Exp/Cntr=0.3,0.1

Type RM Length L Ch R = 1,89164,909,909,909
BEGIN DESCRIPTION:
Elizabeth Creek 100.0
END DESCRIPTION:
XS GIS Cut Line= 4
      2301377.75      7066276.91      2300451.87      7066176.06
      2299946.90      7065984.69      2299002.68      7066116.88
#Sta/Elev= 30
  3306.7  802.85  4019.6  798.61  4489.4  797.63  4578.8  798.07  4584.2  795.31
  4609.0  790.44  4887.0  794.63  4923.4  792.67  4957.7  793.97  4977.9  791.07
  5018.3  789.92  5029.7  787.84  5031.7  787.34  5047.2  787.84  5048.6  789.95
  5058.7  789.56  5078.9  791.75  5137.7  793.35  5169.8  792.22  5209.1  795.42
  5214.1  792.34  5230.3  794.49  5280.5  795.08  5472.7  804.05  5499.7  806.43
  5504.8  805.46  5538.7  808.73  5571.1  810.69  5628.5  811.21  5731.5  811.77
#Mann=6,-1,0
  3306.7    0.05       0  4489.4    0.12       0  5029.7    0.07       0
  5047.2    0.12       0  5538.7    0.05       0  5628.5    0.12       0
Bank Sta=5029.7,5047.2
Exp/Cntr=0.3,0.1

Type RM Length L Ch R = 1,88255,421,421,421
BEGIN DESCRIPTION:
Elizabeth Creek 99.0
END DESCRIPTION:
XS GIS Cut Line= 5
      2302160.27      7066180.73      2301696.77      7065537.62
      2301371.56      7065543.43      2300432.29      7065719.93
      2299013.92      7065877.53
#Sta/Elev= 30
  2872.8  806.76  3533.3  794.09  3619.2  793.04  3654.8  794.49  3733.3  791.59
  4161.5  791.44  4649.4  793.49  4776.9  792.24  4848.1  794.24  4864.5  793.03
  4869.6  794.40  4909.4  792.04  4929.5  791.65  4988.7  787.12  5021.6  786.51
  5023.6  786.01  5039.1  786.51  5040.4  787.82  5060.5  792.41  5100.7  792.24
  5151.0  794.19  5275.7  792.86  5541.3  795.56  5718.2  798.36  5887.3  805.07
  5984.8  810.39  5989.8  809.08  6137.1  816.27  6237.7  818.88  6373.6  820.05
#Mann=7,-1,0
  2872.8    0.05       0  4909.4    0.12       0  5021.6    0.07       0
  5039.1    0.05       0  5275.7    0.05       0  5541.3    0.12       0
  5887.3    0.05       0
Bank Sta=5021.6,5039.1
Exp/Cntr=0.3,0.1

Type RM Length L Ch R = 1,87834,532,532,532
BEGIN DESCRIPTION:
Elizabeth Creek 98.0
END DESCRIPTION:
XS GIS Cut Line= 4
      2302336.86      7066303.38      2301775.24      7065509.21
      2300629.00      7065460.00      2300379.00      7065110.00
#Sta/Elev= 30
  2880.4  812.60  3154.0  804.35  3161.3  806.89  3167.4  805.07  3182.2  803.84
  3283.1  801.12  3785.4  792.60  3821.0  794.90  3849.5  791.86  3939.4  792.23
  4079.5  790.43  4600.0  791.47  4680.1  790.01  4884.5  794.12  4912.1  793.35
  4980.4  788.50  4989.1  784.03  4991.1  783.53  5006.6  784.03  5028.6  784.18
  5049.5  790.41  5079.0  791.71  5158.9  791.71  5209.3  787.58  5244.9  788.32
  5344.5  796.91  5375.1  800.87  5402.2  803.54  5423.1  810.39  5430.5  810.70
#Mann=5,-1,0
  2880.4    0.05       0  4912.1    0.12       0  4989.1    0.07       0
  5006.6    0.12       0  5375.1    0.05       0
Bank Sta=4989.1,5006.6
Exp/Cntr=0.3,0.1

Type RM Length L Ch R = 1,87302,542,542,542
BEGIN DESCRIPTION:
Elizabeth Creek 97.0
END DESCRIPTION:
XS GIS Cut Line= 4
      2302182.36      7065871.75      2301860.71      7065488.54
      2300729.00      7065010.00      2300278.98      7064809.99
#Sta/Elev= 30
  3275.3  799.64  3633.6  794.32  3690.8  792.45  3711.6  792.52  3733.7  794.62
  3768.8  792.06  4059.8  789.39  4295.7  789.59  4354.0  788.41  4430.5  790.27
  4689.5  792.52  4713.0  791.11  4743.8  788.49  4906.6  789.49  4937.0  786.87
  5007.1  785.65  5009.9  782.32  5011.9  781.82  5027.5  782.32  5042.0  790.00
  5077.4  792.37  5117.2  796.10  5135.0  804.00  5140.4  804.10  5146.6  807.89
  5157.5  809.93  5435.9  810.88  5453.0  812.78  5487.9  821.40  5496.8  821.75
#Mann=5,-1,0
  3275.3    0.05       0  4713.0    0.12       0  5009.9    0.07       0
  5027.5    0.12       0  5077.4    0.05       0
Bank Sta=5009.9,5027.5
Exp/Cntr=0.3,0.1

Type RM Length L Ch R = 1,86760,573,573,573
BEGIN DESCRIPTION:
Elizabeth Creek 96.0
END DESCRIPTION:
XS GIS Cut Line= 4
      2302465.43      7065918.73      2302030.82      7065502.70
      2301129.00      7064760.00      2300929.01      7064360.03
#Sta/Elev= 30
  3229.4  801.11  3805.9  792.76  3827.2  793.34  3829.4  794.35  3855.9  794.17
  3862.3  792.95  3919.7  790.33  3962.7  789.66  3969.2  790.50  3997.9  789.11
  4104.8  789.95  4438.3  787.48  4566.0  789.61  4850.1  790.39  4870.9  788.82
  4942.6  787.38  4949.1  786.63  4963.5  782.40  4983.3  780.84  4985.3  780.34
  5000.9  780.84  5002.1  783.00  5013.3  786.28  5044.0  787.51  5097.1  786.70
  5125.1  791.19  5222.9  802.17  5387.8  810.91  5438.1  816.94  5446.5  817.00
#Mann=3,-1,0
  3229.4    0.05       0  4983.3   0.033       0  5000.9    0.05       0
Bank Sta=4983.3,5000.9
Exp/Cntr=0.3,0.1

Type RM Length L Ch R = 1,86187,531,531,531
BEGIN DESCRIPTION:
Elizabeth Creek 95.0
END DESCRIPTION:
XS GIS Cut Line= 3
      2302348.64      7065436.26      2301579.00      7064560.00
      2301129.00      7064260.00
#Sta/Elev= 30
  3834.4  794.09  3853.0  792.33  3937.5  790.74  4228.7  789.43  4540.0  785.74
  4703.2  786.80  4717.4  785.97  4724.1  786.86  4809.5  784.65  4858.8  787.26
  4917.8  786.00  4958.4  784.01  4993.6  784.67  4997.3  781.83  5003.7  781.83
  5014.4  777.71  5016.4  777.21  5032.0  777.71  5059.3  779.02  5065.3  781.79
  5080.3  782.26  5095.3  785.04  5101.3  787.13  5161.0  793.17  5302.6  802.03
  5505.4  810.39  5513.0  811.03  5519.0  813.74  5528.0  815.47  5541.5  816.97
#Mann=5,-1,0
  3834.4    0.05       0  4917.8    0.12       0  5014.4    0.07       0
  5032.0    0.12       0  5161.0    0.05       0
Bank Sta=5014.4,5032
Exp/Cntr=0.3,0.1

Type RM Length L Ch R = 1,85656,1608,1608,1608
BEGIN DESCRIPTION:
Elizabeth Creek 94.0
END DESCRIPTION:
XS GIS Cut Line= 3
      2303829.00      7066760.00      2302029.00      7064360.00
      2301229.00      7063860.00
#Sta/Elev= 30
  2003.9  835.06  2482.0  821.12  2940.4  812.51  3461.2  798.36  3490.4  799.65
  3496.6  801.62  3582.0  801.68  3611.2  795.82  3625.8  795.44  3725.8  794.00
  3746.6  795.45  3811.2  792.69  4117.4  791.48  4175.8  788.86  4617.4  784.98
  4746.6  780.73  4770.6  782.73  4811.2  784.39  4890.4  783.87  4946.6  782.13
  4967.0  778.72  4969.0  778.22  4984.6  778.72  4996.6  779.16  5000.8  783.55
  5034.4  785.82  5098.2  784.69  5273.4  793.40  5708.5  805.91  5947.3  808.62
#Mann=5,-1,0
  2003.9    0.05       0  4770.6    0.12       0  4967.0    0.07       0
  4984.6    0.12       0  5034.4    0.05       0
Bank Sta=4967,4984.6
Exp/Cntr=0.3,0.1

Type RM Length L Ch R = 1,84048,1119,1119,1119
BEGIN DESCRIPTION:
Elizabeth Creek 93.0
END DESCRIPTION:
XS GIS Cut Line= 3
      2304028.98      7064859.98      2303229.00      7064060.00
      2301628.95      7063809.99
#Sta/Elev= 30
  3868.9  803.66  4081.0  795.69  4335.6  788.91  4918.6  782.19  4929.5  781.37
  4957.8  775.27  4963.1  770.55  4965.1  770.05  4980.9  770.55  5002.8  771.03
  5010.4  773.90  5020.5  775.54  5071.1  777.83  5131.8  776.12  5164.7  778.83
  5202.7  779.45  5212.8  778.34  5227.5  773.86  5253.3  777.16  5290.2  779.14
  5334.2  779.39  5344.4  780.85  5365.3  779.78  5614.1  782.37  5780.6  782.34
  5851.6  781.82  6022.5  784.05  6204.7  792.29  6392.4  795.49  6619.7  801.84
#Mann=7,-1,0
  3868.9    0.05       0  4918.6    0.12       0  4963.1    0.07       0
  4980.9    0.12       0  5365.3    0.05       0  5780.6    0.12       0
  5851.6    0.05       0
Bank Sta=4963.1,4980.9
Exp/Cntr=0.3,0.1

Type RM Length L Ch R = 1,82929,542,542,542
BEGIN DESCRIPTION:
Elizabeth Creek 92.0
END DESCRIPTION:
XS GIS Cut Line= 3
      2304379.02      7064760.02      2302979.00      7063210.00
      2302579.00      7063010.00
#Sta/Elev= 30
  2911.3  804.36  2989.4  804.05  3017.8  803.01  3038.7  803.52  3428.1  790.65
  3619.4  787.56  3668.7  785.85  3796.5  783.97  4178.4  781.16  4469.0  776.66
  4554.2  776.66  4589.4  775.61  4631.5  776.72  4667.1  777.52  4773.2  774.57
  4844.2  775.63  4929.4  773.87  4934.5  766.71  4936.5  766.21  4952.6  766.71
  4986.1  769.97  5002.8  769.09  5053.1  770.98  5067.1  770.16  5089.4  771.91
  5124.9  777.78  5142.5  781.26  5187.3  785.28  5380.1  796.97  5447.2  802.52
#Mann=5,-1,0
  2911.3    0.05       0  4631.5    0.12       0  4934.5    0.07       0
  4952.6    0.12       0  5124.9    0.05       0
Bank Sta=4934.5,4952.6
Exp/Cntr=0.3,0.1

Type RM Length L Ch R = 1,82387,1193,1193,1193
BEGIN DESCRIPTION:
Elizabeth Creek 91.0
END DESCRIPTION:
XS GIS Cut Line= 3
      2304779.01      7063960.00      2303379.00      7062860.00
      2302578.96      7062359.98
#Sta/Elev= 30
  3224.7  802.35  3523.9  791.03  4401.9  774.89  4478.2  772.84  4542.4  774.16
  4598.5  771.55  4648.3  772.64  4763.5  776.01  4898.5  774.92  4927.2  771.97
  4954.6  766.40  4969.0  765.53  4974.4  761.36  4976.4  760.86  4992.5  761.36
  4997.9  767.64  5002.0  768.93  5018.7  768.91  5055.3  773.06  5192.0  775.43
  5505.7  782.37  5600.1  786.07  5694.4  792.61  5715.7  798.38  5731.0  799.43
  5736.9  801.74  5913.2  802.89  5925.6  805.61  5935.0  810.48  5948.6  811.98
#Mann=7,-1,0
  3224.7    0.05       0  4401.9    0.12       0  4648.3    0.05       0
  4927.2    0.12       0  4974.4    0.07       0  4992.5    0.12       0
  5192.0    0.05       0
Bank Sta=4974.4,4992.5
Exp/Cntr=0.3,0.1

Type RM Length L Ch R = 1,81194,1097,1097,1097
BEGIN DESCRIPTION:
Elizabeth Creek 90.0
END DESCRIPTION:
XS GIS Cut Line= 4
      2305065.55      7062744.52      2304296.52      7062088.95
      2303218.57      7062007.00      2302638.61      7062038.52
#Sta/Elev= 30
  3615.7  785.68  3829.4  783.11  3900.2  783.68  3942.5  781.91  4091.8  779.86
  4559.5  779.16  4609.8  778.01  4633.8  775.18  4673.6  774.93  4683.9  772.79
  4733.1  769.71  4904.5  768.58  4914.6  768.16  4940.9  763.45  4964.7  762.07
  4984.8  763.54  5004.8  762.84  5015.8  759.53  5017.8  759.03  5034.0  759.53
  5045.0  768.13  5077.1  769.51  5285.6  768.66  5334.4  769.41  5396.0  773.10
  5533.6  776.95  5696.8  781.54  6035.6  797.66  6237.6  804.86  6288.1  808.31
#Mann=5,-1,0
  3615.7    0.05       0  4733.1    0.12       0  5015.8    0.07       0
  5034.0    0.12       0  5533.6    0.05       0
Bank Sta=5015.8,5034
Exp/Cntr=0.3,0.1

Type RM Length L Ch R = 1,80097,272,272,272
BEGIN DESCRIPTION:
Elizabeth Creek 89.0
END DESCRIPTION:
XS GIS Cut Line= 4
      2305216.83      7061969.15      2304673.33      7061597.62
      2304109.09      7061566.56      2303016.83      7061653.99
#Sta/Elev= 30
  4346.4  775.83  4436.1  776.45  4636.3  773.82  4776.4  774.29  4797.4  771.77
  4833.3  771.10  4920.0  772.72  4949.4  770.98  4964.9  766.42  4985.7  761.62
  4991.8  758.42  4995.1  754.66  4997.1  754.16  5013.5  754.66  5019.1  755.51
  5029.1  761.38  5039.1  762.10  5175.5  763.38  5289.5  763.34  5339.6  761.46
  5349.6  763.16  5369.6  761.53  5420.5  768.18  5815.0  772.08  5858.1  772.82
  6176.9  781.32  6272.2  781.64  6304.8  780.06  6603.2  796.35  6665.6  802.90
#Mann=9,-1,0
  4346.4    0.05       0  4436.1   0.075       0  4636.3    0.05       0
  4964.9    0.12       0  4995.1    0.07       0  5013.5    0.12       0
  5175.5    0.05       0  5815.0    0.12       0  5858.1    0.05       0
Bank Sta=4995.1,5013.5
Exp/Cntr=0.3,0.1

Type RM Length L Ch R = 1,79825,777,777,777
BEGIN DESCRIPTION:
Elizabeth Creek 88.0
END DESCRIPTION:
XS GIS Cut Line= 3
      2305292.51      7061887.22      2304907.98      7061445.96
      2304178.99      7060859.99
#Sta/Elev= 30
  4333.0  776.51  4376.1  774.37  4451.4  773.51  4489.0  771.72  4531.8  773.80
  4723.5  770.85  4865.0  770.93  4893.5  767.30  4979.2  765.88  4992.1  763.82
  5000.0  761.79  5006.8  756.17  5019.6  755.08  5021.6  754.58  5038.0  755.08
  5043.2  759.02  5064.0  762.20  5113.6  762.18  5135.1  759.15  5148.8  761.37
  5185.6  761.16  5250.7  764.70  5313.6  766.90  5540.8  769.77  5668.8  775.15
  5712.0  777.99  5725.3  779.82  5732.8  783.13  5747.2  784.82  5853.6  793.55
#Mann=6,-1,0
  4333.0   0.075       0  4451.4    0.05       0  4992.1    0.12       0
  5019.6    0.07       0  5038.0    0.12       0  5250.7    0.05       0
Bank Sta=5019.6,5038
Exp/Cntr=0.3,0.1

Type RM Length L Ch R = 1,79048,550,550,550
BEGIN DESCRIPTION:
Elizabeth Creek 87.0
END DESCRIPTION:
XS GIS Cut Line= 3
      2305429.00      7062360.02      2305079.00      7060810.00
      2304878.98      7060459.96
#Sta/Elev= 30
  3410.7  780.80  3824.6  774.98  3882.3  777.07  3989.7  773.64  4015.6  772.11
  4056.6  773.97  4189.9  771.94  4405.1  765.40  4540.2  763.28  4640.9  760.79
  4657.8  759.25  4662.9  756.64  4671.7  755.85  4692.2  759.81  4754.4  761.76
  4866.5  760.52  4897.2  758.36  4927.2  759.31  4969.0  757.89  4997.2  754.19
  5013.4  755.47  5022.8  754.64  5025.8  751.95  5027.8  751.45  5044.2  751.95
  5045.1  754.16  5057.3  760.23  5080.4  765.21  5264.6  775.12  5402.9  789.41
#Mann=6,-1,0
  3410.7    0.05       0  3824.6   0.075       0  3989.7    0.05       0
  4540.2    0.12       0  5025.8    0.07       0  5044.2    0.05       0
Bank Sta=5025.8,5044.2
Exp/Cntr=0.3,0.1

Type RM Length L Ch R = 1,78498,582,582,582
BEGIN DESCRIPTION:
Elizabeth Creek 86.0
END DESCRIPTION:
XS GIS Cut Line= 3
      2305579.00      7062409.96      2305529.00      7060860.00
      2305079.03      7060360.04
#Sta/Elev= 30
  3449.3  783.61  3631.2  779.08  3859.5  775.84  3959.5  777.76  4159.6  772.41
  4587.8  766.49  4609.9  762.23  4850.0  762.36  4990.1  755.93  5003.4  754.32
  5006.8  751.63  5013.9  753.38  5026.4  749.97  5028.4  749.47  5044.8  749.97
  5049.8  751.81  5084.9  750.68  5092.4  752.91  5127.5  751.71  5155.1  753.86
  5176.8  751.57  5219.4  754.55  5226.9  751.31  5247.8  750.15  5255.3  757.08
  5276.2  762.97  5410.8  765.28  5516.9  772.15  5651.4  785.98  5672.7  793.00
#Mann=7,-1,0
  3449.3    0.05       0  3631.2   0.075       0  4587.8    0.05       0
  5006.8    0.12       0  5026.4   0.033       0  5044.8    0.12       0
  5155.1    0.05       0
Bank Sta=5026.4,5044.8
Exp/Cntr=0.3,0.1

Type RM Length L Ch R = 1,77916,586,586,586
BEGIN DESCRIPTION:
Elizabeth Creek 85.0
END DESCRIPTION:
XS GIS Cut Line= 3
      2306029.00      7061810.00      2305979.00      7060710.00
      2305278.97      7060159.97
#Sta/Elev= 30
  3898.9  777.81  3918.9  777.32  3948.9  772.97  3986.1  774.49  4011.5  771.74
  4089.1  771.98  4099.1  776.61  4109.1  786.28  4129.1  781.34  4149.2  771.76
  4159.2  769.99  4233.7  768.66  4349.4  768.11  4419.4  765.94  4459.5  762.00
  4609.6  759.35  4779.8  760.50  4940.0  758.32  4960.0  756.80  4980.0  750.66
  4998.1  749.07  5000.1  748.57  5016.5  749.07  5028.1  752.09  5106.7  757.61
  5150.0  756.81  5584.7  763.97  5783.6  780.36  5812.5  784.82  5890.3  789.23
#Mann=5,-1,0
  3898.9    0.05       0  3986.1   0.075       0  4233.7    0.05       0
  4998.1   0.033       0  5016.5    0.05       0
Bank Sta=4998.1,5016.5
Exp/Cntr=0.3,0.1

Type RM Length L Ch R = 1,77330,541,541,541
BEGIN DESCRIPTION:
Elizabeth Creek 84.0
END DESCRIPTION:
XS GIS Cut Line= 3
      2306779.01      7061760.03      2306429.00      7060360.00
      2305629.04      7059960.02
#Sta/Elev= 30
  3557.2  777.14  3560.5  776.97  3575.3  774.36  3588.2  774.04  3876.8  768.87
  4021.1  768.53  4077.9  766.04  4330.3  763.92  4441.1  761.74  4606.0  761.76
  4711.7  758.52  4917.9  756.81  4935.9  756.10  4959.1  752.03  4960.2  749.02
  4962.2  748.52  4978.6  749.02  5003.1  749.33  5014.3  752.72  5036.7  754.30
  5089.8  753.42  5156.8  754.44  5201.6  753.01  5268.6  755.52  5394.4  755.58
  5500.6  759.61  5662.8  761.74  5760.6  767.23  5813.7  772.44  5894.7  776.77
#Mann=3,-1,0
  3557.2     0.1       0  3560.5   0.075       0  4077.9    0.05       0
Bank Sta=4960.2,4978.6
Exp/Cntr=0.3,0.1

Type RM Length L Ch R = 1,76789,1674,1674,1674
BEGIN DESCRIPTION:
Elizabeth Creek 83.0
END DESCRIPTION:
XS GIS Cut Line= 3
      2307629.01      7062360.02      2306629.00      7059960.00
      2305764.51      7059398.62
#Sta/Elev= 30
  2400.0  789.61  2438.5  786.64  2881.1  780.84  2898.4  776.66  2934.6  778.72
  2995.9  774.73  3073.7  775.60  3112.3  770.14  3165.4  771.75  3180.0  774.93
  3194.6  784.72  3205.7  786.57  3218.5  788.86  3223.9  795.38  3255.9  784.95
  3348.5  768.64  3523.7  766.08  3560.8  767.87  3584.6  764.69  3762.3  762.19
  4986.9  751.18  5003.2  749.42  5004.5  746.18  5006.5  745.68  5022.9  746.18
  5042.4  746.67  5064.4  753.19  5131.1  753.19  5384.3  753.32  6030.8  774.74
#Mann=7,-1,0
  2400.0    0.05       0  2881.1   0.075       0  3073.7    0.05       0
  3205.7   0.075       0  3523.7    0.05       0  4986.9    0.12       0
  5131.1    0.05       0
Bank Sta=5004.5,5022.9
Exp/Cntr=0.3,0.1

Type RM Length L Ch R = 1,75115,561,561,561
BEGIN DESCRIPTION:
Elizabeth Creek 82.0
END DESCRIPTION:
XS GIS Cut Line= 3
      2308479.01      7061410.02      2307829.00      7059860.00
      2306829.03      7059010.02
#Sta/Elev= 30
  3314.5  774.38  3659.9  762.79  3878.4  756.93  4485.6  750.88  4756.7  749.65
  4874.8  746.69  4956.9  746.91  4973.6  744.94  4980.7  742.44  4986.1  742.47
  4992.6  740.46  5007.5  740.44  5009.5  739.94  5018.1  739.94  5026.0  740.44
  5031.0  743.21  5037.6  744.15  5059.6  742.10  5066.1  742.86  5073.8  746.07
  5497.0  750.51  5556.0  751.10  5662.5  754.52  5683.4  756.17  5754.8  757.64
  5775.6  759.31  5789.9  757.63  5804.2  757.75  6023.8  763.19  6307.7  766.30
#Mann=3,-1,0
  3314.5    0.05       0  5018.1    0.12       0  5497.0    0.05       0
Bank Sta=5007.5,5026
Exp/Cntr=0.3,0.1

Type RM Length L Ch R = 1,74554,828,828,828
BEGIN DESCRIPTION:
Elizabeth Creek 81.0
END DESCRIPTION:
XS GIS Cut Line= 3
      2308579.00      7061059.98      2308229.00      7059510.00
      2307428.96      7059259.99
#Sta/Elev= 30
  3410.7  765.70  3492.7  764.30  3544.0  761.13  3759.2  760.07  3769.5  759.80
  3795.9  756.32  3839.1  755.12  4162.0  750.15  4474.7  747.80  4662.9  748.08
  4754.4  746.54  4804.9  744.64  4923.0  744.05  4938.2  742.93  4948.4  738.80
  4958.7  736.98  4987.8  736.44  4989.8  735.94  5006.4  736.44  5015.9  738.61
  5053.7  743.15  5062.6  741.64  5086.1  742.51  5135.9  741.07  5183.6  746.07
  5209.2  746.91  5247.2  749.97  5324.5  753.80  5471.2  758.42  5837.9  761.64
#Mann=5,-1,0
  3410.7    0.05       0  4923.0    0.12       0  4987.8    0.07       0
  5006.4    0.12       0  5247.2    0.05       0
Bank Sta=4987.8,5006.4
Exp/Cntr=0.3,0.1

Type RM Length L Ch R = 1,73726,404,404,404
BEGIN DESCRIPTION:
Elizabeth Creek 80.5
END DESCRIPTION:
XS GIS Cut Line= 3
      2309043.28      7060449.98      2308721.78      7059138.78
      2308255.27      7058955.95
#Sta/Elev= 30
  4287.1  756.10  4441.5  755.11  4678.3  748.45  4745.6  747.26  4833.9  743.88
  4863.7  743.45  4925.4  744.64  4966.6  744.42  4976.9  744.02  4987.2  741.80
  4995.2  738.03  5000.3  737.18  5008.8  731.67  5010.8  731.17  5027.4  731.67
  5028.4  736.46  5036.7  736.01  5041.9  737.09  5049.0  733.97  5057.4  736.00
  5069.6  738.07  5083.5  738.41  5100.5  740.89  5152.0  740.47  5193.1  743.21
  5252.8  744.50  5849.0  748.71  6041.0  750.27  6110.4  750.24  6138.2  751.08
#Mann=7,-1,0
  4287.1    0.05       0  5008.8    0.05       0  5027.4    0.05       0
  5057.4    0.12       0  5252.8    0.05       0  5849.0    0.12       0
  6041.0    0.05       0
Bank Sta=5008.8,5027.4
Exp/Cntr=0.3,0.1

Type RM Length L Ch R = 1,73322,957,957,957
BEGIN DESCRIPTION:
Elizabeth Creek 80.2
END DESCRIPTION:
XS GIS Cut Line= 3
      2309314.34      7060412.17      2309219.78      7059277.46
      2309276.51      7058521.02
#Sta/Elev= 30
  4270.7  755.17  4583.9  753.13  4814.7  749.13  4878.4  746.15  4935.2  740.07
  4965.3  738.21  4975.3  736.01  4989.5  730.87  4991.5  730.37  5008.1  730.87
  5015.4  734.35  5045.5  737.60  5125.8  735.50  5196.1  742.07  5371.7  742.82
  5409.3  742.92  5416.8  741.87  5426.8  736.10  5436.9  734.12  5446.9  736.51
  5497.0  735.30  5567.2  742.23  5687.6  747.67  5747.7  752.60  5787.9  760.82
  5838.0  768.01  5878.1  770.20  5888.1  769.69  5958.3  774.15  6167.9  781.00
#Mann=4,-1,0
  4270.7    0.05       0  4989.5   0.033       0  5008.1    0.05       0
  5371.7    0.05       0
Bank Sta=4989.5,5008.1
Exp/Cntr=0.3,0.1

Type RM Length L Ch R = 1,72365,572,572,572
BEGIN DESCRIPTION:
Elizabeth Creek 80.0
END DESCRIPTION:
XS GIS Cut Line= 3
      2309478.97      7060260.03      2310029.00      7059660.00
      2309879.00      7058860.02
#Sta/Elev= 30
  4186.1  752.98  4490.4  748.28  4596.5  744.77  4724.1  738.40  4853.1  738.17
  4922.1  737.57  4950.4  734.85  4964.6  734.48  4978.8  732.69  4986.2  728.62
  4998.6  727.69  5001.0  727.19  5021.9  727.69  5026.4  728.76  5040.8  728.06
  5051.0  730.70  5061.1  736.40  5071.3  738.74  5084.0  739.40  5136.6  737.76
  5173.0  739.01  5189.2  738.52  5265.1  739.77  5447.7  743.21  5529.1  743.19
  5671.6  744.79  5782.7  749.68  5787.7  750.03  5803.8  753.51  5814.0  754.49
#Mann=5,-1,0
  4186.1    0.05       0  4853.1    0.12       0  4998.6    0.07       0
  5021.9    0.12       0  5265.1    0.05       0
Bank Sta=4998.6,5021.9
Exp/Cntr=0.3,0.1

Type RM Length L Ch R = 1,71793,546,546,546
BEGIN DESCRIPTION:
Elizabeth Creek 79.0
END DESCRIPTION:
XS GIS Cut Line= 3
      2309978.99      7060810.02      2310529.00      7059560.00
      2311328.97      7058760.03
#Sta/Elev= 30
  3634.3  754.89  3968.5  747.48  4126.0  748.07  4166.2  743.02  4195.0  742.38
  4212.9  743.99  4235.2  742.66  4241.7  746.33  4265.0  750.00  4270.5  749.65
  4282.2  742.59  4300.8  737.77  4439.3  735.35  4453.7  733.46  4520.3  736.64
  4741.2  737.70  4879.8  735.32  4938.9  736.34  4975.4  732.40  4991.0  731.47
  4997.2  728.14  5016.3  727.17  5018.7  726.67  5040.2  727.17  5084.8  736.79
  5127.3  735.85  5396.0  739.99  5692.9  747.85  5989.9  764.00  6131.3  777.11
#Mann=5,-1,0
  3634.3    0.05       0  4282.2    0.12       0  4975.4    0.05       0
  5016.3    0.07       0  5040.2    0.05       0
Bank Sta=5016.3,5040.2
Exp/Cntr=0.3,0.1

Type RM Length L Ch R = 1,71247,527,527,527
BEGIN DESCRIPTION:
Elizabeth Creek 78.0
END DESCRIPTION:
XS GIS Cut Line= 3
      2310228.98      7060610.02      2310929.00      7059810.00
      2311428.98      7059010.03
#Sta/Elev= 30
  3937.0  751.29  4007.7  749.50  4036.2  751.84  4043.3  748.34  4057.1  747.59
  4078.9  751.48  4099.8  747.10  4121.6  750.60  4142.5  745.11  4149.6  747.06
  4185.2  743.48  4282.4  742.87  4291.5  743.55  4305.8  737.86  4334.2  731.77
  4418.7  735.97  4536.3  736.11  4829.7  733.34  4872.4  736.53  4960.1  723.99
  4962.5  723.49  4984.0  723.99  5007.7  726.46  5028.9  733.46  5107.9  732.11
  5181.1  737.36  5412.8  735.94  5558.4  740.80  5878.0  760.05  5943.4  767.40
#Mann=5,-1,0
  3937.0    0.05       0  4282.4    0.12       0  4536.3    0.05       0
  4960.1    0.05       0  4984.0    0.05       0
Bank Sta=4960.1,4984
Exp/Cntr=0.3,0.1

Type RM Length L Ch R = 1,70720,548,548,548
BEGIN DESCRIPTION:
Elizabeth Creek 77.0
END DESCRIPTION:
XS GIS Cut Line= 3
      2310678.99      7060660.01      2311379.00      7059910.00
      2311479.01      7059109.96
#Sta/Elev= 30
  3968.7  747.54  4258.7  742.13  4280.2  736.97  4287.0  737.65  4294.3  732.85
  4322.7  730.17  4365.2  733.78  4393.0  730.79  4478.0  732.45  4556.2  729.72
  4739.9  735.85  4782.4  733.33  4860.0  734.49  4888.4  732.75  4895.7  729.71
  4945.0  729.11  4952.4  725.72  4959.2  728.55  4966.5  723.27  4979.2  722.07
  4981.6  721.57  5003.2  722.07  5024.9  723.42  5032.4  726.62  5037.5  723.46
  5045.0  726.81  5176.0  732.18  5458.2  733.27  5619.5  747.85  5800.9  758.91
#Mann=3,-1,0
  3968.7    0.05       0  4979.2   0.033       0  5003.2    0.05       0
Bank Sta=4979.2,5003.2
Exp/Cntr=0.3,0.1

Type RM Length L Ch R = 1,70172,566,566,566
BEGIN DESCRIPTION:
Elizabeth Creek 76.0
END DESCRIPTION:
XS GIS Cut Line= 3
      2311579.00      7061560.02      2311779.00      7059560.00
      2311679.00      7059060.00
#Sta/Elev= 30
  2994.5  757.54  3024.7  756.93  3054.8  753.60  3074.9  755.74  3142.8  754.38
  3617.6  737.42  3637.7  738.35  3677.9  736.18  3868.9  733.18  4059.8  731.23
  4449.2  733.11  4783.4  729.76  4823.6  733.51  4833.6  733.06  4851.2  727.36
  4856.3  728.96  4883.9  720.62  4956.8  721.41  4962.3  719.29  4964.7  718.79
  4986.3  719.29  4994.4  725.44  5002.0  727.59  5188.1  728.14  5231.5  732.95
  5266.8  743.54  5279.8  748.06  5310.4  750.89  5392.0  754.35  5514.4  763.08
#Mann=5,-1,0
  2994.5    0.05       0  4962.3   0.033       0  4986.3    0.05       0
  5231.5    0.12       0  5266.8    0.05       0
Bank Sta=4962.3,4986.3
Exp/Cntr=0.3,0.1

Type RM Length L Ch R = 1,69606,589,589,589
BEGIN DESCRIPTION:
Elizabeth Creek 75.0
END DESCRIPTION:
XS GIS Cut Line= 3
      2311528.99      7061810.04      2312329.00      7059610.00
      2311879.01      7058860.02
#Sta/Elev= 30
  2663.3  759.47  2759.1  758.11  2780.4  753.71  2821.0  757.41  2887.5  754.66
  2943.3  757.16  2993.2  753.30  3014.5  755.35  3116.2  753.03  3553.8  737.25
  4022.0  728.52  4397.8  731.05  4693.7  729.10  4802.1  726.02  4841.3  726.47
  4866.0  730.20  4960.4  716.44  4962.8  715.94  4984.4  716.44  4989.0  723.36
  5012.1  728.93  5193.6  727.51  5256.7  726.44  5309.4  725.92  5354.1  724.13
  5398.8  728.90  5426.1  727.80  5484.4  744.23  5509.4  746.23  5878.9  761.27
#Mann=7,-1,0
  2663.3    0.05       0  4960.4   0.033       0  4984.4    0.05       0
  5193.6    0.12       0  5256.7    0.05       0  5309.4    0.12       0
  5509.4    0.05       0
Bank Sta=4960.4,4984.4
Exp/Cntr=0.3,0.1

Type RM Length L Ch R = 1,69017,530,530,530
BEGIN DESCRIPTION:
Elizabeth Creek 74.0
END DESCRIPTION:
XS GIS Cut Line= 3
      2311779.02      7061359.98      2312779.00      7059960.00
      2312978.98      7059610.04
#Sta/Elev= 30
  3274.9  751.05  3383.0  745.69  3798.4  734.89  4379.7  726.35  4614.4  727.72
  4709.0  726.89  4820.3  724.14  4836.8  724.95  4860.2  724.13  4872.4  726.05
  4895.8  726.83  4937.6  720.93  4967.1  718.86  4973.2  717.85  4980.1  713.45
  4982.6  712.95  5004.4  713.45  5009.0  714.10  5024.8  721.13  5030.6  722.79
  5040.7  723.39  5089.6  722.69  5121.3  720.85  5133.5  718.48  5142.9  721.26
  5170.3  725.60  5201.9  728.24  5219.3  730.74  5309.9  740.52  5398.4  745.92
#Mann=5,-1,0
  3274.9    0.05       0  4820.3    0.12       0  4980.1    0.07       0
  5004.4    0.12       0  5219.3    0.05       0
Bank Sta=4980.1,5004.4
Exp/Cntr=0.3,0.1

Type RM Length L Ch R = 1,68487,319,319,319
BEGIN DESCRIPTION:
Elizabeth Creek 73.0
END DESCRIPTION:
XS GIS Cut Line= 3
      2311878.97      7061460.03      2313029.00      7060360.00
      2313228.99      7059610.03
#Sta/Elev= 30
  3409.1  751.93  3550.5  746.04  3939.5  735.92  4703.5  727.09  4908.5  723.72
  4929.9  723.75  4939.5  724.91  4972.4  722.80  4986.5  718.61  4993.4  715.26
  5010.9  714.38  5013.4  713.88  5035.4  714.38  5041.9  717.27  5073.0  719.84
  5098.2  724.27  5114.4  724.32  5145.4  721.56  5213.3  721.97  5280.0  720.08
  5321.4  720.96  5352.4  723.55  5373.7  727.74  5411.1  731.80  5476.6  732.57
  5569.7  735.60  5611.1  739.75  5693.9  741.89  5735.3  748.25  5776.7  749.74
#Mann=5,-1,0
  3409.1    0.05       0  4939.5    0.12       0  5010.9    0.07       0
  5035.4    0.12       0  5411.1    0.05       0
Bank Sta=5010.9,5035.4
Exp/Cntr=0.3,0.1

Type RM Length L Ch R = 1,68168,87,87,87
BEGIN DESCRIPTION:
Elizabeth Creek 72.2
END DESCRIPTION:
XS GIS Cut Line= 2
      2313292.17      7061555.44      2313355.07      7059630.47
#Sta/Elev= 30
  3853.6  731.64  3899.1  730.14  3911.8  729.04  3929.1  725.65  3959.1  727.78
  4249.2  729.96  4539.4  727.62  4809.5  724.25  4879.6  723.92  4909.6  724.87
  4919.6  721.07  4929.6  718.62  4969.6  715.25  4977.4  713.90  4979.8  713.40
  5001.9  713.90  5009.7  717.28  5026.2  718.73  5037.8  720.45  5059.7  721.28
  5129.6  720.07  5319.8  723.42  5359.8  725.17  5459.9  732.26  5499.9  733.11
  5519.9  735.44  5539.9  736.40  5620.0  743.08  5640.0  745.83  5779.6  749.43
#Mann=5,-1,0
  3853.6    0.05       0  4977.4   0.033       0  5001.9    0.05       0
  5026.2    0.12       0  5037.8    0.05       0
Bank Sta=4977.4,5001.9
Exp/Cntr=0.3,0.1

Type RM Length L Ch R = 1,68081,822,822,822
BEGIN DESCRIPTION:
Elizabeth Creek 72.3
END DESCRIPTION:
XS GIS Cut Line= 2
      2313397.96      7061520.16      2313411.80      7059838.51
#Sta/Elev= 30
  3917.8  731.16  3948.0  729.64  3978.0  725.73  4078.0  726.84  4168.0  728.91
  4308.0  729.71  4518.0  728.11  4568.0  727.04  4608.0  727.62  4638.0  726.73
  4768.0  725.11  4888.0  724.64  4938.0  723.10  4968.0  716.80  4995.7  714.18
  4998.2  713.68  5017.8  713.68  5020.2  714.18  5028.0  715.45  5058.0  717.83
  5078.0  723.72  5088.0  724.28  5218.0  722.18  5288.0  722.66  5308.0  723.70
  5348.0  724.10  5378.0  725.67  5468.0  732.79  5518.0  735.79  5599.5  739.09
#Mann=3,-1,0
  3917.8    0.05       0  4995.7   0.033       0  5020.2    0.05       0
Bank Sta=4995.7,5020.2
Exp/Cntr=0.3,0.1

Type RM Length L Ch R = 1,67259,726,726,726
BEGIN DESCRIPTION:
Elizabeth Creek 72.4
END DESCRIPTION:
XS GIS Cut Line= 4
      2313471.21      7061528.23      2313586.77      7060846.17
      2314098.91      7060418.45      2314080.01      7059844.90
#Sta/Elev= 30
  3418.7  731.90  3438.8  731.19  3467.6  723.76  3711.0  728.15  4066.0  727.29
  4436.3  722.04  4796.2  720.46  4846.2  719.09  4866.2  715.46  4916.3  713.27
  4924.1  713.71  4929.1  715.77  4936.3  714.79  4975.5  713.91  4986.3  712.10
  4994.1  709.36  4996.5  708.86  5018.6  709.36  5026.3  712.29  5036.3  718.26
  5046.3  718.79  5096.4  716.60  5146.4  716.51  5176.4  715.31  5206.4  715.79
  5266.5  723.08  5290.4  728.73  5306.5  734.31  5326.5  737.03  5351.6  738.64
#Mann=5,-1,0
  3418.7    0.05       0  4975.5    0.12       0  4994.1    0.07       0
  5018.6    0.12       0  5290.4    0.05       0
Bank Sta=4994.1,5018.6
Exp/Cntr=0.3,0.1

Type RM Length L Ch R = 1,66533,252,252,252
BEGIN DESCRIPTION:
Elizabeth Creek 72.5
END DESCRIPTION:
XS GIS Cut Line= 4
      2313498.32      7061517.45      2313647.51      7060836.59
      2314622.13      7060260.85      2314842.42      7059864.32
#Sta/Elev= 30
  2944.5  731.98  2952.1  731.90  2982.8  723.70  2993.1  723.49  3203.8  727.80
  3641.5  726.23  4062.3  719.29  4493.5  717.39  4524.8  714.99  4543.6  711.16
  4560.8  709.76  4573.5  714.36  4589.1  717.10  4816.5  717.88  4911.7  714.90
  4925.2  712.26  4946.9  713.22  4957.2  709.27  4984.7  711.01  4991.8  710.64
  4994.1  708.67  4996.6  708.17  5018.7  708.67  5028.1  717.42  5049.9  729.81
  5060.2  734.45  5082.6  739.27  5087.6  742.60  5109.4  745.49  5227.1  751.75
#Mann=5,-1,0
  2944.5    0.05       0  4543.6    0.12       0  4994.1    0.07       0
  5018.7    0.12       0  5082.6    0.05       0
Bank Sta=4994.1,5018.7
Exp/Cntr=0.3,0.1

Type RM Length L Ch R = 1,66281,575,575,575
BEGIN DESCRIPTION:
Elizabeth Creek 72.0
END DESCRIPTION:
XS GIS Cut Line= 4
      2313571.57      7061547.25      2313683.89      7060863.12
      2314929.00      7060210.00      2315328.99      7060160.00
#Sta/Elev= 30
  2904.9  732.79  2942.6  732.07  2984.9  722.81  3256.8  726.39  3597.2  725.68
  3700.9  721.87  3728.6  723.09  3739.3  720.50  3773.3  721.80  3899.4  719.35
  4152.7  719.38  4454.1  716.34  4500.0  714.69  4544.1  710.21  4560.5  710.90
  4575.1  716.62  4781.1  716.81  4913.9  712.86  4946.2  714.05  4968.3  710.73
  4973.9  706.01  4983.7  704.67  4986.1  704.17  5008.3  704.67  5014.3  711.91
  5054.6  738.42  5074.7  746.57  5098.0  749.47  5236.0  754.71  5407.3  755.00
#Mann=5,-1,0
  2904.9    0.05       0  4454.1    0.12       0  4983.7    0.07       0
  5008.3    0.12       0  5098.0    0.05       0
Bank Sta=4983.7,5008.3
Exp/Cntr=0.3,0.1

Type RM Length L Ch R = 1,65706,554,554,554
BEGIN DESCRIPTION:
Elizabeth Creek 71.0
END DESCRIPTION:
XS GIS Cut Line= 3
      2313929.00      7061510.00      2314929.00      7060710.00
      2315229.01      7060409.99
#Sta/Elev= 30
  3719.5  731.35  3755.5  727.37  3761.9  723.94  3797.1  722.49  4090.1  723.45
  4480.7  719.68  4515.9  725.89  4538.3  722.10  4559.1  723.31  4643.9  716.86
  4680.0  723.32  4730.4  714.44  4751.2  714.89  4765.6  717.69  4772.0  722.28
  4794.4  723.79  4815.2  722.20  4822.8  715.37  4908.1  712.84  4943.3  704.35
  4959.6  703.74  4962.1  703.24  4984.6  703.74  5028.4  711.16  5155.7  711.68
  5226.4  707.87  5240.5  710.46  5303.0  741.52  5339.5  751.12  5424.4  754.13
#Mann=5,-1,0
  3719.5    0.05       0  4822.8    0.12       0  4959.6    0.07       0
  4984.6    0.12       0  5303.0    0.05       0
Bank Sta=4959.6,4984.6
Exp/Cntr=0.3,0.1

Type RM Length L Ch R = 1,65152,533,533,533
BEGIN DESCRIPTION:
Elizabeth Creek 70.0
END DESCRIPTION:
XS GIS Cut Line= 3
      2314078.97      7061610.01      2315229.00      7061110.00
      2315229.00      7060510.03
#Sta/Elev= 30
  3741.0  730.30  3795.6  729.56  3817.4  727.91  3878.2  727.52  3883.6  728.42
  4000.8  726.02  4100.1  721.90  4175.8  723.52  4373.5  720.95  4591.6  716.45
  4654.0  717.26  4955.0  716.66  4973.2  712.68  4980.6  709.10  4986.0  703.81
  4997.5  705.15  5002.5  702.60  5005.0  702.10  5027.5  702.60  5065.0  706.80
  5105.0  709.72  5225.0  710.44  5312.9  712.42  5375.0  714.78  5405.4  718.89
  5425.0  722.40  5445.0  728.50  5506.4  740.34  5535.0  747.71  5595.0  752.84
#Mann=7,-1,0
  3741.0    0.05       0  4955.0    0.12       0  5002.5    0.07       0
  5027.5    0.12       0  5312.9    0.05       0  5405.4    0.12       0
  5506.4    0.05       0
Bank Sta=5002.5,5027.5
Exp/Cntr=0.3,0.1

Type RM Length L Ch R = 1,64619,1081,1081,1081
BEGIN DESCRIPTION:
Elizabeth Creek 69.0
END DESCRIPTION:
XS GIS Cut Line= 3
      2315542.49      7061559.40      2315729.00      7061110.00
      2315611.85      7060254.75
#Sta/Elev= 30
  4509.4  721.24  4537.6  719.54  4620.1  718.57  4627.8  716.45  4649.5  714.85
  4660.3  718.04  4682.0  718.40  4909.7  715.96  4928.2  712.29  4933.6  712.96
  4952.0  706.52  4957.5  707.71  4963.5  704.38  4977.3  703.04  4993.6  700.47
  4996.1  699.97  5018.6  700.47  5046.4  705.15  5066.6  706.89  5127.2  705.98
  5187.7  711.76  5232.1  711.14  5369.4  712.75  5541.0  721.06  5619.5  730.36
  5624.6  729.77  5682.3  740.82  5696.7  741.19  5753.0  747.89  5859.2  750.97
#Mann=5,-1,0
  4509.4    0.05       0  4977.3    0.12       0  4993.6    0.07       0
  5018.6    0.12       0  5232.1    0.05       0
Bank Sta=4993.6,5018.6
Exp/Cntr=0.3,0.1

Type RM Length L Ch R = 1,63538,566,566,566
BEGIN DESCRIPTION:
Elizabeth Creek 68.0
END DESCRIPTION:
XS GIS Cut Line= 3
      2316532.18      7061685.51      2316329.00      7060310.00
      2315929.04      7060260.01
#Sta/Elev= 30
  3613.6  719.70  3841.6  717.82  3861.8  713.76  3875.9  714.09  3882.0  716.44
  4094.9  714.09  4162.5  713.61  4316.7  710.89  4326.8  710.32  4347.0  703.71
  4353.0  703.48  4375.5  705.92  4556.7  709.43  4913.1  704.83  4933.3  703.90
  4953.5  697.29  4961.8  696.38  4964.3  695.88  4986.8  696.38  5001.5  707.95
  5014.1  709.77  5041.8  718.07  5046.9  723.64  5054.4  725.59  5095.8  728.25
  5114.9  729.96  5135.0  736.46  5215.7  743.38  5306.4  747.47  5407.1  747.37
#Mann=7,-1,0
  3613.6    0.05       0  4094.9    0.12       0  4162.5    0.05       0
  4375.5    0.12       0  4961.8    0.07       0  4986.8    0.12       0
  5095.8    0.05       0
Bank Sta=4961.8,4986.8
Exp/Cntr=0.3,0.1

Type RM Length L Ch R = 1,62972,645,645,645
BEGIN DESCRIPTION:
Elizabeth Creek 67.0
END DESCRIPTION:
XS GIS Cut Line= 3
      2317004.96      7061597.29      2316879.00      7060260.00
      2316529.02      7060010.02
#Sta/Elev= 30
  3656.9  718.57  3704.4  719.53  3744.6  717.47  3824.9  717.05  3835.0  714.88
  3845.0  714.67  4100.3  712.48  4391.8  711.16  4658.6  709.44  4786.2  704.27
  4837.3  702.48  4869.5  704.95  4959.9  703.07  4970.0  702.23  4980.0  698.24
  4990.1  696.36  5009.7  695.80  5012.2  695.30  5034.7  695.80  5037.0  698.63
  5049.3  700.10  5114.4  699.28  5143.9  697.10  5179.5  701.58  5185.7  703.52
  5194.3  703.17  5242.1  707.01  5307.3  714.96  5344.2  717.70  5430.2  720.92
#Mann=7,-1,0
  3656.9    0.05       0  4100.3    0.12       0  4391.8    0.05       0
  4786.2    0.12       0  5009.7    0.07       0  5034.7    0.12       0
  5242.1    0.05       0
Bank Sta=5009.7,5034.7
Exp/Cntr=0.3,0.1

Type RM Length L Ch R = 1,62327,997,997,997
BEGIN DESCRIPTION:
Elizabeth Creek 66.0
END DESCRIPTION:
XS GIS Cut Line= 3
      2317490.35      7060966.88      2317402.10      7059977.18
      2317219.51      7059234.21
#Sta/Elev= 30
  3988.9  711.22  4357.2  709.12  4518.1  707.07  4588.1  704.87  4688.5  704.84
  4843.2  701.74  4909.4  698.95  4929.5  696.05  4982.5  694.13  4987.7  692.29
  4990.2  691.79  5012.7  692.29  5016.1  697.59  5041.4  701.78  5057.6  699.77
  5104.3  702.57  5187.4  702.09  5216.5  698.43  5228.9  697.91  5237.1  701.15
  5247.4  702.51  5265.3  701.63  5312.0  701.90  5431.5  705.54  5436.7  704.66
  5537.5  710.53  5556.2  712.00  5566.6  714.51  5679.9  721.79  5747.6  728.18
#Mann=6,-1,0
  3988.9    0.12       0  4518.1    0.05       0  4843.2    0.12       0
  4987.7    0.07       0  5012.7    0.12       0  5537.5    0.05       0
Bank Sta=4987.7,5012.7
Exp/Cntr=0.3,0.1

Type RM Length L Ch R = 1,61330,640,640,640
BEGIN DESCRIPTION:
Elizabeth Creek 65.5
END DESCRIPTION:
XS GIS Cut Line= 4
      2317484.05      7061143.38      2318026.18      7060368.01
      2318183.77      7059636.77      2318032.62      7058824.33
#Sta/Elev= 30
  3236.5  712.66  3280.7  712.39  3530.2  711.37  3686.2  709.36  4171.9  706.39
  4174.1  706.33  4446.5  704.19  4553.0  701.90  4569.3  701.00  4589.7  698.02
  4597.2  694.88  4605.5  694.80  4610.2  693.64  4640.9  696.88  4740.0  698.52
  4906.9  697.70  4947.7  697.06  4957.9  694.03  4988.7  689.53  5016.6  689.47
  5019.1  688.97  5041.6  689.47  5049.4  695.78  5059.6  695.96  5100.3  701.48
  5137.1  703.76  5531.6  720.92  5589.5  724.09  5637.2  728.32  5757.0  732.58
#Mann=9,-1,0
  3236.5    0.05       0  3280.7    0.12       0  3686.2    0.05       0
  4171.9    0.12       0  4174.1    0.05       0  4605.5    0.12       0
  5016.6    0.07       0  5041.6    0.12       0  5137.1    0.05       0
Bank Sta=5016.6,5041.6
Exp/Cntr=0.3,0.1

Type RM Length L Ch R = 1,60690,452,452,452
BEGIN DESCRIPTION:
Elizabeth Creek 65.2
END DESCRIPTION:
XS GIS Cut Line= 3
      2318675.47      7061080.37      2318549.39      7059548.52
      2318183.90      7058918.37
#Sta/Elev= 30
  3775.4  710.51  3852.1  709.72  4417.0  704.52  4749.6  698.86  4869.5  699.21
  4892.5  698.16  4959.8  693.03  4969.8  687.98  4977.4  687.91  4979.9  687.41
  5002.4  687.91  5020.0  692.80  5140.4  697.50  5256.0  696.07  5280.8  693.82
  5290.9  691.85  5300.9  692.09  5306.4  693.83  5333.8  696.62  5341.4  698.44
  5384.4  699.91  5421.7  703.16  5459.0  703.03  5495.7  704.52  5507.8  703.83
  5743.0  712.87  5882.1  721.14  5919.4  725.95  5940.9  727.37  6040.9  732.32
#Mann=7,-1,0
  3775.4    0.05       0  3852.1    0.12       0  4417.0    0.05       0
  4749.6    0.12       0  4977.4    0.07       0  5002.4    0.12       0
  5306.4    0.05       0
Bank Sta=4977.4,5002.4
Exp/Cntr=0.3,0.1

Type RM Length L Ch R = 1,60238,545,545,545
BEGIN DESCRIPTION:
Elizabeth Creek 65.0
END DESCRIPTION:
XS GIS Cut Line= 3
      2319179.00      7061010.01      2318979.00      7059910.00
      2318428.98      7059109.98
#Sta/Elev= 30
  3889.9  714.36  3975.0  712.70  4150.8  705.96  4645.9  701.57  4845.3  696.21
  4875.8  697.15  4927.9  696.05  4953.3  692.31  4967.3  688.18  4985.3  687.64
  4987.8  687.14  5010.3  687.64  5015.4  690.42  5021.5  688.64  5030.3  694.13
  5123.0  695.14  5215.6  693.39  5266.4  695.22  5281.3  693.74  5353.0  693.95
  5359.9  689.32  5373.9  689.73  5403.7  696.63  5415.0  696.73  5481.5  697.62
  5526.2  701.76  5748.2  705.24  5857.4  708.57  5935.5  712.32  5978.8  716.09
#Mann=7,-1,0
  3889.9    0.05       0  4150.8    0.12       0  4645.9    0.05       0
  4953.3    0.12       0  4985.3    0.07       0  5010.3    0.12       0
  5415.0    0.05       0
Bank Sta=4985.3,5010.3
Exp/Cntr=0.3,0.1

Type RM Length L Ch R = 1,59693,562,562,562
BEGIN DESCRIPTION:
Elizabeth Creek 64.0
END DESCRIPTION:
XS GIS Cut Line= 3
      2319229.01      7061009.97      2319479.00      7059910.00
      2319229.00      7058310.03
#Sta/Elev= 30
  3867.7  714.98  4031.7  708.98  4146.9  706.57  4267.6  703.94  4477.3  703.10
  4525.5  701.43  4743.5  699.73  4903.4  695.72  4976.7  697.26  4985.5  695.77
  4993.2  688.82  4998.2  688.82  5005.8  685.59  5023.7  685.03  5026.2  684.53
  5048.7  685.03  5056.4  691.63  5076.7  692.74  5147.5  690.85  5188.0  693.07
  5238.6  691.31  5279.1  692.03  5319.6  689.57  5360.1  692.99  5428.1  694.82
  5996.2  706.49  6098.9  711.84  6200.2  720.14  6432.9  730.50  6615.1  740.83
#Mann=6,-1,0
  3867.7    0.05       0  4146.9    0.12       0  4743.5    0.05       0
  5023.7   0.033       0  5048.7    0.05       0  5428.1    0.05       0
Bank Sta=5023.7,5048.7
Exp/Cntr=0.3,0.1

Type RM Length L Ch R = 1,59131,563,563,563
BEGIN DESCRIPTION:
Elizabeth Creek 63.0
END DESCRIPTION:
XS GIS Cut Line= 3
      2320428.98      7060409.97      2319929.00      7059610.00
      2319479.02      7058810.04
#Sta/Elev= 30
  4060.8  720.02  4083.8  719.44  4126.2  713.46  4199.3  707.71  4280.9  704.95
  4357.3  700.50  4480.0  699.30  4499.4  699.37  4606.2  698.96  4857.2  695.96
  4874.4  696.72  4917.5  687.56  4959.9  688.10  4975.3  684.77  4988.7  684.48
  4991.2  683.98  5013.7  684.48  5017.9  684.61  5027.1  691.58  5084.5  691.15
  5130.4  686.84  5196.9  689.92  5260.7  690.81  5276.7  694.88  5291.0  695.31
  5313.9  691.86  5341.7  695.93  5590.3  696.84  5724.8  699.72  5922.0  710.41
#Mann=9,-1,0
  4060.8    0.05       0  4280.9    0.12       0  4480.0   0.075       0
  4499.4    0.12       0  4606.2    0.05       0  4857.2    0.12       0
  4988.7    0.07       0  5013.7    0.12       0  5196.9    0.05       0
Bank Sta=4988.7,5013.7
Exp/Cntr=0.3,0.1

Type RM Length L Ch R = 1,58568,587,587,587
BEGIN DESCRIPTION:
Elizabeth Creek 62.0
END DESCRIPTION:
XS GIS Cut Line= 3
      2320479.00      7060509.96      2320429.00      7059410.00
      2319628.97      7058609.97
#Sta/Elev= 30
  3894.1  715.65  3924.1  717.51  3984.1  715.55  3994.2  712.97  4001.7  708.92
  4006.7  715.67  4014.2  712.01  4034.2  710.03  4217.4  702.31  4503.6  697.74
  4556.1  697.14  4654.1  696.21  4887.6  692.67  4945.1  690.01  4955.1  688.74
  4962.7  684.51  4965.2  684.01  4987.7  684.51  5008.1  685.35  5051.8  688.11
  5065.9  687.00  5080.0  689.08  5122.5  687.37  5155.1  688.41  5207.3  688.80
  5292.2  694.35  5730.6  696.27  5872.0  698.73  5971.0  702.30  6126.6  713.84
#Mann=9,-1,0
  3894.1    0.05       0  4217.4    0.12       0  4503.6    0.05       0
  4556.1    0.12       0  4654.1    0.05       0  4962.7   0.033       0
  4987.7    0.05       0  5008.1    0.12       0  5155.1    0.05       0
Bank Sta=4962.7,4987.7
Exp/Cntr=0.3,0.1

Type RM Length L Ch R = 1,57981,363,363,363
BEGIN DESCRIPTION:
Elizabeth Creek 61.0
END DESCRIPTION:
XS GIS Cut Line= 3
      2322041.66      7060367.98      2320829.00      7059010.00
      2320132.93      7058226.18
#Sta/Elev= 30
  3184.3  703.33  3333.3  702.10  3369.3  700.60  3390.2  697.35  3425.3  700.68
  3496.4  701.53  3843.3  696.78  4120.0  688.93  4126.7  690.21  4487.9  691.00
  4544.7  689.82  4601.5  691.10  4687.7  685.75  4690.2  685.25  4712.7  685.75
  4969.4  687.28  5026.2  690.28  5111.5  690.55  5160.9  693.11  5175.1  691.46
  5181.8  693.94  5189.3  691.89  5210.2  693.70  5245.7  691.14  5330.6  690.94
  5685.2  695.96  5826.6  702.57  5897.6  711.05  5926.1  716.54  6053.2  725.95
#Mann=3,-1,0
  3184.3    0.05       0  4687.7   0.033       0  4712.7    0.05       0
Bank Sta=4687.7,4712.7
Exp/Cntr=0.3,0.1

Type RM Length L Ch R = 1,57618,709,709,709
BEGIN DESCRIPTION:
Elizabeth Creek 60.0
END DESCRIPTION:
XS GIS Cut Line= 3
      2322533.41      7060374.34      2321064.60      7058773.16
      2320686.42      7057934.84
#Sta/Elev= 30
  2934.4  706.73  3442.8  697.49  4030.4  692.62  4356.0  686.06  4610.7  687.17
  4759.3  685.72  4766.7  683.58  4773.5  685.64  4780.9  683.36  4787.6  685.77
  4844.4  685.80  4851.8  683.73  4858.5  685.96  4865.9  683.83  4901.1  686.03
  4915.3  682.76  4922.1  686.36  4929.5  683.30  4936.2  685.67  4964.6  684.52
  4973.7  680.92  4976.2  680.42  4998.7  680.92  5028.7  680.92  5092.2  687.28
  5417.9  690.48  5620.1  696.49  5769.8  713.90  5954.9  726.78  6026.9  734.61
#Mann=3,-1,0
  2934.4    0.05       0  4973.7   0.033       0  4998.7    0.05       0
Bank Sta=4973.7,4998.7
Exp/Cntr=0.3,0.1

Type RM Length L Ch R = 1,56909,1099,1099,1099
BEGIN DESCRIPTION:
Elizabeth Creek 59.0
END DESCRIPTION:
XS GIS Cut Line= 3
      2322646.83      7060122.14      2321729.00      7058810.00
      2321078.98      7058009.97
#Sta/Elev= 30
  3399.2  703.99  3499.4  702.75  3706.9  695.74  4764.2  684.60  4878.5  685.32
  4921.6  682.30  4963.9  683.01  4972.1  676.21  4984.9  676.18  4987.4  675.68
  5009.9  676.18  5050.8  678.76  5064.9  677.40  5071.6  680.09  5078.0  676.97
  5135.5  682.00  5149.9  678.64  5156.3  681.16  5164.3  679.24  5220.3  679.36
  5228.2  684.89  5275.6  685.66  5335.2  687.18  5455.2  685.77  5498.3  689.29
  5797.1  689.82  5817.9  694.96  5875.4  697.98  5966.8  707.74  6031.3  711.88
#Mann=5,-1,0
  3399.2    0.05       0  4764.2    0.12       0  4984.9    0.07       0
  5009.9    0.12       0  5275.6    0.05       0
Bank Sta=4984.9,5009.9
Exp/Cntr=0.3,0.1

Type RM Length L Ch R = 1,55810,568,568,568
BEGIN DESCRIPTION:
Elizabeth Creek 58.0
END DESCRIPTION:
XS GIS Cut Line= 3
      2323478.99      7059659.99      2322679.00      7058410.00
      2321078.99      7057710.00
#Sta/Elev= 30
  3512.4  704.70  3783.6  695.12  3853.4  693.51  4807.1  683.13  4873.8  679.58
  4910.2  681.38  4925.0  677.89  4931.4  680.20  4952.5  675.18  4970.4  673.53
  4972.9  673.03  4995.4  673.53  5018.3  674.58  5028.8  679.58  5034.3  678.14
  5051.0  680.72  5109.9  678.99  5149.3  680.62  5203.5  678.45  5269.3  682.04
  5313.4  681.08  5382.1  683.06  5552.8  682.25  5680.6  678.07  5738.7  681.50
  6204.5  690.04  6355.8  695.88  6501.6  708.42  6681.7  717.23  6742.9  722.55
#Mann=7,-1,0
  3512.4    0.05       0  3783.6    0.12       0  3853.4    0.05       0
  4925.0    0.12       0  4970.4    0.07       0  4995.4    0.12       0
  5382.1    0.05       0
Bank Sta=4970.4,4995.4
Exp/Cntr=0.3,0.1

Type RM Length L Ch R = 1,55242,570,570,570
BEGIN DESCRIPTION:
Elizabeth Creek 57.0
END DESCRIPTION:
XS GIS Cut Line= 3
      2323529.00      7059559.99      2322879.00      7058010.00
      2321879.03      7057460.02
#Sta/Elev= 30
  3313.9  703.07  3449.2  697.48  3505.7  694.76  3556.4  694.27  3736.0  690.97
  4366.2  685.94  4506.7  683.35  4528.4  681.18  4550.1  676.88  4560.8  676.45
  4643.9  680.27  4744.4  681.32  4842.9  680.78  4956.3  678.99  4973.0  675.46
  4985.5  676.67  5008.4  671.65  5027.8  670.58  5030.3  670.08  5052.8  670.58
  5062.4  678.01  5068.1  679.83  5111.6  681.76  5302.8  677.66  5399.6  680.37
  5589.9  680.25  5930.5  688.58  5997.2  691.66  6113.1  701.80  6135.9  702.52
#Mann=6,-1,0
  3313.9    0.05       0  3449.2    0.12       0  3556.4    0.05       0
  4560.8    0.12       0  5027.8    0.07       0  5052.8    0.05       0
Bank Sta=5027.8,5052.8
Exp/Cntr=0.3,0.1

Type RM Length L Ch R = 1,54672,544,544,544
BEGIN DESCRIPTION:
Elizabeth Creek 56.0
END DESCRIPTION:
XS GIS Cut Line= 3
      2323729.01      7059460.05      2323379.00      7057910.00
      2322078.96      7057209.98
#Sta/Elev= 30
  3405.8  700.89  3528.9  697.60  3580.1  694.36  3704.6  691.96  4482.3  684.34
  4686.5  678.70  4749.6  672.71  4759.1  675.75  4787.6  677.70  4975.8  678.82
  4984.6  677.79  4992.3  668.48  5012.4  667.76  5014.9  667.26  5037.4  667.76
  5090.6  672.29  5106.8  671.68  5112.5  674.60  5128.7  673.92  5156.3  675.76
  5172.5  675.29  5178.2  677.81  5264.6  680.34  5533.5  677.34  5880.8  679.41
  6073.8  683.22  6266.1  689.06  6337.5  692.80  6413.8  700.26  6471.4  702.03
#Mann=5,-1,0
  3405.8    0.05       0  4686.5    0.12       0  5012.4    0.07       0
  5037.4    0.12       0  5264.6    0.05       0
Bank Sta=5012.4,5037.4
Exp/Cntr=0.3,0.1
