--- Farris Branch.prj (project) ---

Proj Title=Farris Branch Base Level Engineering
Current Plan=p01
Default Exp/Contr=0.3,0.1
English Units
Geom File=g01
Flow File=f01
Plan File=p01
Y Axis Title=Elevation
X Axis Title(PF)=Main Channel Distance
X Axis Title(XS)=Station
BEGIN DESCRIPTION:
Farris Branch
END DESCRIPTION:
DSS Export Rating Curves= 0
DSS Export Rating Curve Sorted= 0
DSS Export Volume Flow Curves= 0
DXF OffsetX= 0
DXF OffsetY= 0
DXF ScaleX= 1
DXF ScaleY= 10

--- Farris Branch.p01 (plan) ---

Plan Title=Multiple Run
Program Version=4.10
Short Identifier=Multiple
Geom File=g01
Flow File=f01
Subcritical Flow
K Sum by GR= 0
Std Step Tol= 0.01
Critical Tol= 0.01
Num of Std Step Trials= 20
Max Error Tol= 0.3
Flow Tol Ratio= 0.001
Split Flow NTrial= 30
Split Flow Tol= 0.02
Split Flow Ratio= 0.02
Log Output Level= 0
Friction Slope Method= 1
Unsteady Friction Slope Method= 2
Unsteady Bridges Friction Slope Method= 1
Parabolic Critical Depth
Global Vel Dist= 1 , 1 , 1
Global Log Level= 0
CheckData=True
Encroach Param=-1 ,0,0, 0
BEGIN DESCRIPTION:
Multiple Run
END DESCRIPTION:
Computation Interval=1HOUR
Output Interval=1HOUR
Run HTab= 0
Run UNet= 0
Run PostProcess= 0
Run WQNet= 0
UNET Theta= 1
UNET Theta Warmup= 1
UNET ZTol= 0.02
UNET ZSATol= 0.05
UNET MxIter= 20
UNET MaxInSteps= 0
UNET DtIC= 0
UNET DtMin= 0
UNET MaxCRTS= 20
UNET WFStab= 2
UNET SFStab= 1
UNET WFX= 1
UNET SFX= 1
UNET DSS MLevel= 4
UNET DZMax Abort= 100
UNET Convert EG Bridges= 0
UNET Use Existing IB Tables=-1
UNET Froude Reduction=False
UNET Froude Limit= 1
UNET Froude Power= 10
UNET Time Slicing=0,0, 5
UNET Junction Losses=0
Instantaneous Interval=1HOUR
Write IC File= 0
Write IC File at Sim End=0
Echo Input=False
Echo Parameters=False
Echo Output=False
Write Detailed= 0
WQ AD Non Conservative
WQ ULTIMATE=-1
WQ Max Comp Step=1HOUR
WQ Output Interval=15MIN
WQ Output Selected Increments= 0
WQ Output face flow=0
WQ Output face velocity=0
WQ Output face area=0
WQ Output face dispersion=0
WQ Output cell volume=0
WQ Output cell surface area=0
WQ Output cell continuity=0
WQ Output cumulative cell continuity=0
WQ Output face conc=0
WQ Output face dconc_dx=0
WQ Output face courant=0
WQ Output face peclet=0
WQ Output face adv mass=0
WQ Output face disp mass=0
WQ Output cell mass=0
WQ Output cell source sink temp=0
WQ Output cell source sink nsm=0
WQ Output MaxMinRange=-1
WQ Daily Max Min Mean=-1
WQ Daily Range=0
WQ Daily Time=0
WQ Create Restart=0
WQ Fixed Restart=0
WQ System Summary=0
WQ Use Fixed Temperature=0
Sorting and Armoring Iterations= 10
XS Update Threshold= 0.02
Hydraulics Update Threshold= 0.02
Energy Slope Method= 1
Volume Change Method= 0
XS Weighting Method= 0
Number of US Weighted Cross Sections= 1
Number of DS Weighted Cross Sections= 1
Upstream XS Weight=0.25
Main XS Weight=0.5
Downstream XS Weight=0.25
Number of DS XS's Weighted with US Boundary= 1
Upstream Boundary Weight= 1
Weight of XSs Associated with US Boundary= 0
Number of US XS's Weighted with DS Boundary= 1
Downstream Boundary Weight= 0.5
Weight of XSs Associated with DS Boundary= 0.5
Sediment Output Level= 4
Mass or Volume Output= 0
Output Increment Type= 1
Profile and TS Output Increment= 10
XS Output Flag= 0
XS Output Increment= 10
Disregard all LS=0
Disregard all Conn=0
Disregard all Breaches=0
Disregard all Pumps=0

--- Farris Branch.f01 (steady flow) ---

Flow Title=Multiple
Number of Profiles=7
Profile Names=10-year,25-year,50-year,1pct_min,100-year,1pct_plu,500-year
River Rch & RM= Farris Branch,Reach-1,20889
     354     470     564     336     671    1340     949
River Rch & RM= Farris Branch,Reach-1,16752
     721     993    1219     742    1480    2953    2181
River Rch & RM= Farris Branch,Reach-1,11243
     910    1271    1574     965    1925    3842    2883
River Rch & RM= Farris Branch,Reach-1,9941
    1021    1434    1782    1097    2189    4367    3301
River Rch & RM= Farris Branch,Reach-1,8957
    1469    2099    2638    1640    3272    6528    5034
River Rch & RM= Farris Branch,Reach-1,6338
    1803    2597    3281    2048    4085    8151    6341
River Rch & RM= Farris Branch,Reach-1,3699
    1899    2740    3465    2164    4317    8613    6709
Boundary for River Rch & Prof#=Farris Branch,Reach-1,1
Up Type=0
Dn Type=3
Dn Slope=0.005
Boundary for River Rch & Prof#=Farris Branch,Reach-1,2
Up Type=0
Dn Type=3
Dn Slope=0.005
Boundary for River Rch & Prof#=Farris Branch,Reach-1,3
Up Type=0
Dn Type=3
Dn Slope=0.005
Boundary for River Rch & Prof#=Farris Branch,Reach-1,4
Up Type=0
Dn Type=3
Dn Slope=0.005
Boundary for River Rch & Prof#=Farris Branch,Reach-1,5
Up Type=0
Dn Type=3
Dn Slope=0.005
Boundary for River Rch & Prof#=Farris Branch,Reach-1,6
Up Type=0
Dn Type=3
Dn Slope=0.005
Boundary for River Rch & Prof#=Farris Branch,Reach-1,7
Up Type=0
Dn Type=3
Dn Slope=0.005

--- Farris Branch.g01 (geometry) ---

Geom Title=Existing Conditions
Program Version=4.10

River Reach=Farris Branch   ,Reach-1
Reach XY= 30
        2398979.        7026060.      2399180.09      7027699.46
      2399436.86      7028366.17      2399980.55      7028806.25
      2400523.14      7028812.05        2400879.        7029010.
      2400931.07      7029704.16      2401129.87      7029854.89
      2400880.08      7030670.55      2400886.65       7031213.7
      2401173.94       7031357.7      2401111.68      7031593.73
      2401326.09      7031617.91      2401378.06      7032049.52
      2401179.98      7032348.31      2401388.83      7032370.47
      2401484.18      7032654.56      2401773.75      7032807.35
        2401579.        7033060.      2401732.35      7033301.91
      2402799.03      7033609.94      2403285.26      7033361.95
      2403681.74      7033415.34      2403981.06      7034754.15
      2404158.84      7034940.37        2404679.        7034960.
      2405922.95      7036001.84      2406849.09      7036379.79
        2408479.        7038510.        2408179.        7039410.

Type RM Length L Ch R = 1 ,20889   ,43,43,43
BEGIN DESCRIPTION:
Farris Branch 47.0
END DESCRIPTION:
XS GIS Cut Line= 4
      2398799.16      7026447.78      2398879.83      7026313.33
      2399054.58      7026254.18      2399232.03      7026192.34
#Sta/Elev= 30
  4738.9  643.93  4840.5  643.13  4846.3  642.71  4889.1  641.92  4897.9  642.22
  4915.9  641.59  4921.4  641.91  4947.6  639.45  4956.2  636.74  4956.4  636.24
  4959.9  636.24  4960.2  636.74  4984.3  637.55  4989.8  636.81  5000.4  637.25
  5010.5  639.25  5032.1  646.51  5041.9  647.12  5047.2  650.34  5053.2  647.24
  5063.7  645.94  5073.3   645.8  5078.6  648.86  5085.2  649.63  5095.5  654.66
  5116.6  655.56  5166.6  655.93  5171.9  656.61  5253.5  656.96  5268.1  656.94
#Mann= 4 ,-1 , 0
  4738.9     .05       0  4956.2     .05       0  4960.2     .05       0
  5253.5    .075       0
Bank Sta=4956.2,4960.2
XS Rating Curve= 0 ,0
Exp/Cntr=0.3,0.1

Type RM Length L Ch R = 1 ,20846   ,100,100,100
BEGIN DESCRIPTION:
Farris Branch 46.0
END DESCRIPTION:
XS GIS Cut Line= 4
      2398809.95      7026469.23      2398898.65      7026334.83
      2399062.64      7026310.64      2399265.47       7026219.9
#Sta/Elev= 30
  4757.9  643.79  4872.5  642.79  4939.5  641.37  4979.9  641.89  4985.6  641.11
  5000.1  636.76  5008.3  635.24  5008.5  634.74    5012  634.74  5012.3  635.24
  5020.4  635.37  5030.5  636.82  5040.6  641.35  5050.2  644.09  5060.8  644.83
  5084.7  645.07  5097.8  647.41  5113.6  647.54  5126.5  650.35  5144.2  650.06
  5149.7  652.75  5167.4  652.14  5172.9  653.37  5190.3  652.06  5212.2  652.69
  5224.8   653.9  5242.5  653.93    5248   654.7  5277.9  656.53  5306.9  657.48
#Mann= 3 ,-1 , 0
  4757.9     .05       0  5008.3     .05       0  5012.3     .05       0
Bank Sta=5008.3,5012.3
XS Rating Curve= 0 ,0
Exp/Cntr=0.3,0.1

Type RM Length L Ch R = 1 ,20746   ,253,253,253
BEGIN DESCRIPTION:
Farris Branch 45.0
END DESCRIPTION:
XS GIS Cut Line= 3
      2398817.98      7026490.77      2398960.48      7026423.55
      2399178.28      7026369.77
#Sta/Elev= 30
  4777.6  643.78  4787.7  644.52  4793.2  643.73  4800.8  644.49  4810.5  644.49
  4838.8  643.95  4845.1  642.99  4861.5  643.09  4884.3  641.98  4889.9  642.31
  4907.1  641.69  4954.2  641.59  4964.5  638.95  4970.3  635.98  4993.4  634.33
  4993.7  633.83  4997.2  633.83  4997.4  634.33  5005.7  637.55  5011.7  642.48
  5016.9   642.4  5036.6  645.46  5046.9  648.21  5067.5  649.18  5077.8  647.57
  5094.6  650.06  5099.8  648.71  5108.7  649.63  5136.1  651.04  5159.5  651.66
#Mann= 3 ,-1 , 0
  4777.6     .05       0  4993.4     .05       0  4997.4     .05       0
Bank Sta=4993.4,4997.4
XS Rating Curve= 0 ,0
Exp/Cntr=0.3,0.1

Type RM Length L Ch R = 1 ,20493   ,287,287,287
BEGIN DESCRIPTION:
Farris Branch 44.0
END DESCRIPTION:
XS GIS Cut Line= 3
       2398905.9      7026660.53      2399055.88      7026660.53
       2399154.9      7026660.53
#Sta/Elev= 27
  4876.9  643.97  4880.9  643.97    4890   643.2    4900  642.72    4910  642.15
    4920  641.25    4930  640.84    4950  640.32    4960  639.98    4970  639.93
  4979.9  637.37    4990   634.6    5000  632.65  5008.3  632.05  5011.8  632.05
    5015  632.55    5020  633.71  5030.9  636.29    5040  640.75    5050   643.9
    5060  644.59    5080  644.89    5090  646.16    5100  646.64    5110  646.66
    5120  647.06  5125.9  647.46
#Mann= 4 ,-1 , 0
  4876.9      .1       0  4979.9     .05       0    5000    .045       0
    5015     .05       0
Bank Sta=5000,5015
XS Rating Curve= 0 ,0
Exp/Cntr=0.3,0.1

Type RM Length L Ch R = 1 ,20206   ,150,150,150
BEGIN DESCRIPTION:
Farris Branch 43.0
END DESCRIPTION:
XS GIS Cut Line= 3
      2398906.76       7026920.9      2399135.23      7026934.33
      2399261.62      7026899.38
#Sta/Elev= 30
  4827.5  644.12  4869.8  642.79  4889.8  642.63  4896.1  642.06  4901.1  642.17
  4923.1  637.23  4939.9  633.53    4960  630.99    4968  626.99  4968.2  626.49
  4971.7  626.49    4972  626.99    4980  629.14    4990   630.2    5000  630.53
  5010.1  631.28  5020.1  635.68  5030.1  638.91  5040.1  639.68  5060.9  640.15
  5070.7  640.79    5081  643.11  5088.8  643.04    5094  643.98  5133.5  645.46
  5143.3  645.66  5162.6   645.5  5167.8  645.91  5174.4  646.05  5187.5  645.72
#Mann= 4 ,-1 , 0
  4827.5    .075       0  4923.1     .05       0    4968     .05       0
    4972     .05       0
Bank Sta=4968,4972
XS Rating Curve= 0 ,0
Exp/Cntr=0.3,0.1

Type RM Length L Ch R = 1 ,20056   ,91,91,91
BEGIN DESCRIPTION:
Farris Branch 42.7
END DESCRIPTION:
XS GIS Cut Line= 3
      2398858.29      7027082.19      2399014.25      7027079.51
      2399293.86      7027068.75
#Sta/Elev= 30
  4762.6  640.75  4793.3  637.66  4813.3  637.26  4823.3  637.65  4833.3  639.29
  4843.3  639.73  4853.3  639.27  4873.3   639.3  4893.3   635.2  4913.3  633.77
  4918.5  632.14  4923.5  632.14  4933.3  630.67  4943.4  629.92  4963.4  629.88
  4973.4  628.87  5003.4  628.79  5011.4  623.26  5011.7  622.76  5015.2  622.76
  5015.4  623.26  5023.4  626.49  5032.1  632.03  5037.1  630.65  5043.4  633.51
  5063.4  636.75  5093.5  638.74  5143.5  639.13  5183.5  640.95  5198.4  641.08
#Mann= 3 ,-1 , 0
  4762.6     .05       0  5011.4    .033       0  5015.4     .05       0
Bank Sta=5011.4,5015.4
XS Rating Curve= 0 ,0
Exp/Cntr=0.3,0.1

Type RM Length L Ch R = 1 ,19965   ,164,164,164
BEGIN DESCRIPTION:
Farris Branch 42.5
END DESCRIPTION:
XS GIS Cut Line= 3
      2398874.49      7027162.84      2399030.38      7027160.16
      2399309.96       7027149.4
#Sta/Elev= 30
  4741.9  640.33  4796.4  639.91  4806.4  638.52  4816.4  637.96  4856.4  633.57
  4866.4  631.44  4886.4  629.21  4926.5  627.21  4936.5  625.68  4946.5  625.38
  4956.5  623.25  4966.5   619.5  4974.5  618.03  4974.7  617.53  4978.2  617.53
  4978.5  618.03  4986.5  619.84  4996.5  624.12  5006.5  625.37  5016.5  625.88
  5026.5  625.17  5031.7  625.54  5036.8  629.58  5056.5  631.88  5066.6  632.46
  5076.6  634.13  5106.6  635.96  5116.6  636.09  5136.6     638  5177.6  638.72
#Mann= 3 ,-1 , 0
  4741.9     .05       0  4974.5    .033       0  4978.5     .05       0
Bank Sta=4974.5,4978.5
XS Rating Curve= 0 ,0
Exp/Cntr=0.3,0.1

Type RM Length L Ch R = 1 ,19801   ,220,220,220
BEGIN DESCRIPTION:
Farris Branch 42.0
END DESCRIPTION:
XS GIS Cut Line= 3
      2399029.04        7027310.       2399210.5      7027302.64
      2399404.03      7027262.32
#Sta/Elev= 30
  4847.6  638.76  4867.6  637.85  4877.6   635.2  4887.6  630.53  4897.6  631.45
  4910.3  631.74  4937.6  631.63  4947.6  630.74  4957.7  630.51  4971.8  627.33
  4977.7  623.85  4987.7  620.37  4992.1  619.39  4997.7  618.15  5005.7  617.22
  5005.9  616.72  5009.4  616.72  5009.7  617.22  5017.7  622.68    5026  626.15
  5029.2  626.15  5037.9  629.42  5070.2  635.64  5078.8  635.79  5099.2  637.68
  5120.2  638.75  5160.8  639.14  5165.2  639.73  5180.9  639.32  5226.9  640.99
#Mann= 6 ,-1 , 0
  4847.6      .1       0  4910.3     .05       0  4992.1     .12       0
  5005.7     .07       0  5009.7     .12       0  5160.8     .05       0
Bank Sta=5005.7,5009.7
XS Rating Curve= 0 ,0
Exp/Cntr=0.3,0.1

Type RM Length L Ch R = 1 ,19581   ,285,285,285
BEGIN DESCRIPTION:
Farris Branch 41.0
END DESCRIPTION:
XS GIS Cut Line= 3
      2398925.57      7027445.13      2399172.86      7027509.64
      2399460.54      7027504.26
#Sta/Elev= 30
  4687.9  642.14  4688.6  642.14  4732.8  642.04  4815.5  638.89  4825.8  635.09
  4836.1  626.25  4848.7  625.03  4854.9  625.52  4877.5   626.5  4898.1  626.05
  4918.8   624.1  4924.5   622.6  4929.7  623.66  4943.5  622.97  4959.6   617.1
  4967.6  615.14  4967.9  614.64  4971.6  615.14  4979.6  615.52  4999.6  619.25
  5029.6  619.85  5069.6  622.91  5089.6   623.5  5119.6  629.72  5139.6   632.4
  5146.2  634.68  5149.6  635.86  5159.6   636.3  5169.6  634.25  5231.2  636.44
#Mann= 6 ,-1 , 0
  4687.9      .1       0  4688.6     .05       0  4854.9     .12       0
  4967.6     .07       0  4971.6     .12       0  5146.2     .05       0
Bank Sta=4967.6,4971.6
XS Rating Curve= 0 ,0
Exp/Cntr=0.3,0.1

Type RM Length L Ch R = 1 ,19296   ,249,249,249
BEGIN DESCRIPTION:
Farris Branch 40.0
END DESCRIPTION:
XS GIS Cut Line= 3
       2399062.6      7027826.88        2399229.        7027760.
      2399511.06      7027614.76
#Sta/Elev= 30
  4825.2  633.48  4828.5  632.69  4858.1  631.86  4864.4  630.62  4929.1  624.01
  4941.4  621.79  4950.7  621.12  4965.6  615.48  4972.2  614.11    4988  613.54
  5012.8  614.07  5018.4   617.3    5035  617.84  5040.6  621.59  5049.5  624.51
  5057.2  620.87  5062.8  623.88    5072  625.28  5107.1  623.71  5123.7   624.4
  5129.3  623.55  5171.5  623.55  5201.7  623.99  5228.9   624.9  5234.5  626.66
  5251.1  625.73  5256.7  633.26  5273.2  630.76  5278.9  634.62  5321.8  636.24
#Mann= 5 ,-1 , 0
  4825.2     .12       0  4972.2    .035       0  5012.8     .12       0
  5171.5    .075       0  5201.7     .05       0
Bank Sta=4972.2,5012.8
XS Rating Curve= 0 ,0
Exp/Cntr=0.3,0.1

Type RM Length L Ch R = 1 ,19047   ,155,155,155
BEGIN DESCRIPTION:
Farris Branch 39.0
END DESCRIPTION:
XS GIS Cut Line= 3
       2399057.3      7027974.73      2399369.11       7027980.1
      2399541.17      7027920.96
#Sta/Elev= 30
  4728.8  632.03  4745.1  631.53  4750.5  630.99  4760.5  631.02  4770.5  630.67
  4790.5  630.51  4800.5  629.15  4820.5  627.95  4840.5  625.81  4864.1  623.74
  4870.5  623.36  4880.5  623.17  4890.5  622.64  4910.5  614.54  5028.8  613.46
  5032.3  613.46  5061.7  615.09  5072.3  615.91  5082.3  616.25  5087.6  616.73
  5093.4  616.77    5104  622.76  5113.6  624.23  5118.9  625.64  5199.2  625.45
  5207.3  625.23  5212.6  625.41  5218.8  624.59  5220.5  624.59  5222.6  624.59
#Mann= 5 ,-1 , 0
  4728.8    .075       0  4864.1     .12       0  4910.5    .035       0
  5061.7    .075       0  5220.5      .1       0
Bank Sta=4910.5,5061.7
XS Rating Curve= 0 ,0
Exp/Cntr=0.3,0.1

Type RM Length L Ch R = 1 ,18892   ,176,176,176
BEGIN DESCRIPTION:
Farris Branch 38.3
END DESCRIPTION:
XS GIS Cut Line= 3
      2399031.54      7028137.61      2399449.76      7028114.52
      2399724.56      7028102.95
#Sta/Elev= 30
  4631.8  631.17  4679.3  629.77  4696.7  628.08  4719.4  628.62  4739.4  628.32
  4749.4  627.11  4789.5  625.23  4819.5  624.98  4839.6  624.15  4859.6  624.31
  4877.6  622.73  4882.6  621.74  4889.6  619.35  4929.7  614.05    4978   613.5
  4999.8  614.12  5009.8  614.88  5019.8  616.43  5029.8  620.09  5039.9  622.62
  5058.4  624.63  5063.4  624.23  5067.8  625.55  5119.9  625.18    5150  626.26
    5190  628.71  5219.5  631.37    5230  632.72  5250.1  634.12  5325.7  636.19
#Mann= 4 ,-1 , 0
  4631.8    .075       0  4929.7    .035       0  4999.8    .075       0
  5219.5      .1       0
Bank Sta=4929.7,4999.8
XS Rating Curve= 0 ,0
Exp/Cntr=0.3,0.1

Type RM Length L Ch R = 1 ,18716   ,221,221,221
BEGIN DESCRIPTION:
Farris Branch 38.0
END DESCRIPTION:
XS GIS Cut Line= 3
      2399030.38      7028300.01      2399468.58      7028275.82
      2399723.98      7028265.07
#Sta/Elev= 30
  4601.2  624.85  4639.9  622.38  4669.9  621.54  4688.6  621.31  4693.6  622.47
  4760.1  618.91  4790.1  618.36  4820.2  616.57  4840.2  616.52  4869.4   614.5
  4874.4  616.15  4900.3  615.98  4910.3  615.38  4930.3  612.43  4960.4  603.43
  4968.4  603.31  4968.6  602.81  4972.4  603.31  4980.4  604.59  4990.4  608.57
  5000.4  611.03  5050.5  615.77  5062.5  618.94  5080.5  621.68  5087.2  622.04
  5100.5  623.19  5140.6  624.75  5160.6  626.98  5180.6  628.26  5295.7  629.67
#Mann= 4 ,-1 , 0
  4601.2     .05       0  4968.4     .05       0  4972.4     .05       0
  5087.2    .075       0
Bank Sta=4968.4,4972.4
XS Rating Curve= 0 ,0
Exp/Cntr=0.3,0.1

Type RM Length L Ch R = 1 ,18495   ,259,259,259
BEGIN DESCRIPTION:
Farris Branch 37.0
END DESCRIPTION:
XS GIS Cut Line= 3
      2399279.02      7028709.98        2399529.        7028460.
      2399578.98      7028360.03
#Sta/Elev= 30
  4646.5  624.61  4674.8  623.26    4703  620.49  4712.7  620.47    4802  617.39
  4844.5  614.38  4858.6  613.06  4872.8  609.71  4886.9  608.37    4901  603.32
  4915.2  603.86  4929.3  607.28  4943.5  608.04  4957.6  606.04  4969.7  598.42
    4970  597.92  4973.7  598.42  4974.3  598.63  4985.9   602.6  4996.5  608.06
  5002.8  608.06  5022.4  612.71  5036.4  612.75  5045.9   613.6  5067.1  615.72
  5075.5  617.23  5081.1  617.12  5103.4  620.82    5109  622.78  5111.8  622.78
#Mann= 6 ,-1 , 0
  4646.5     .05       0  4712.7     .12       0  4969.7     .05       0
  4973.7     .12       0  4974.3     .05       0  5045.9    .075       0
Bank Sta=4969.7,4973.7
XS Rating Curve= 0 ,0
Exp/Cntr=0.3,0.1

Type RM Length L Ch R = 1 ,18236   ,267,267,267
BEGIN DESCRIPTION:
Farris Branch 36.0
END DESCRIPTION:
XS GIS Cut Line= 3
      2399578.82      7028899.49      2399683.65      7028657.56
      2399828.98      7028460.03
#Sta/Elev= 30
    4634  622.07  4724.3  618.21  4764.2  615.79  4807.8  612.17  4840.5  611.31
  4852.5   609.8  4893.6  607.84  4914.2  606.26  4920.4   604.6  4928.8  603.85
  4943.5  602.98  4949.7  603.43  4956.7  602.57  4964.3  600.35  4970.5  601.55
  4983.2  596.43  4983.4  595.93  4987.2  596.43  4993.6  598.88  4999.8  599.35
  5006.4  601.94  5014.5  603.93  5020.7  601.76  5029.1  603.61  5035.3   602.9
    5050  605.27  5085.5  608.95  5093.3  621.36  5112.2  622.41  5142.9  623.92
#Mann= 4 ,-1 , 0
    4634     .12       0  4983.2     .07       0  4987.2     .12       0
  5112.2    .075       0
Bank Sta=4983.2,4987.2
XS Rating Curve= 0 ,0
Exp/Cntr=0.3,0.1

Type RM Length L Ch R = 1 ,17969   ,232,232,232
BEGIN DESCRIPTION:
Farris Branch 35.0
END DESCRIPTION:
XS GIS Cut Line= 3
      2399861.07      7028977.52      2399904.09      7028789.29
      2399955.17      7028609.18
#Sta/Elev= 30
  4777.4  617.02  4785.1  617.19  4826.1  615.97  4846.7   614.6  4881.4  610.95
  4902.3  607.43  4918.5  605.83  4924.4  603.92    4939  601.85  4967.3  599.14
  4970.3  600.16  4972.7  600.16  4980.1  599.06  4990.5  596.73  5000.9  593.07
  5004.5  590.92  5004.7  590.42  5008.2  590.42  5008.5  590.92  5011.7  591.58
  5021.7  599.44  5040.4  605.23  5052.9  608.53  5073.7  610.65  5079.5  611.65
  5094.5  612.14  5125.7  614.12  5136.1  615.19  5146.4  617.26  5157.7  615.89
#Mann= 4 ,-1 , 0
  4777.4     .05       0  4902.3     .12       0  5004.5     .07       0
  5008.5     .12       0
Bank Sta=5004.5,5008.5
XS Rating Curve= 0 ,0
Exp/Cntr=0.3,0.1

Type RM Length L Ch R = 1 ,17737   ,292,292,292
BEGIN DESCRIPTION:
Farris Branch 34.0
END DESCRIPTION:
XS GIS Cut Line= 3
      2400121.85      7028942.51        2400129.        7028810.
       2400132.6      7028614.73
#Sta/Elev= 30
  4866.9   605.3  4870.6   605.3  4889.4  603.34  4899.5  602.63  4905.6  601.61
  4939.5  599.16  4947.9  599.31  4959.5   598.7  4969.6  597.82  4979.6   594.6
  4989.6  590.53  4995.1  590.29  4995.3  589.79  4998.8  589.79  4999.1  590.29
  5002.1  590.29  5009.6  590.94  5019.6  592.76  5029.6  593.36  5039.6  598.34
  5049.6   600.9  5059.6  602.28  5069.6  603.35  5079.6  604.81  5089.6  605.35
  5099.6  607.13  5129.6  609.92  5143.5  611.65  5159.6   613.7  5194.9  614.59
#Mann= 5 ,-1 , 0
  4866.9     .05       0  4947.9     .12       0  4995.1     .07       0
  4999.1     .12       0  5143.5      .1       0
Bank Sta=4995.1,4999.1
XS Rating Curve= 0 ,0
Exp/Cntr=0.3,0.1

Type RM Length L Ch R = 1 ,17445   ,114,114,114
BEGIN DESCRIPTION:
Farris Branch 33.0
END DESCRIPTION:
XS GIS Cut Line= 3
      2400350.37      7029025.84      2400390.68      7028869.94
      2400379.98       7028623.8
#Sta/Elev= 30
  4780.5   605.9  4786.5  606.54  4807.2  604.39  4839.1  602.75  4874.6  601.56
  4889.8  600.49  4900.1  599.32  4920.8   598.8  4931.1  597.64  4938.9  593.94
    4944  593.94  4951.5  589.12  4969.5   588.4  4969.7   587.9  4973.2   587.9
  4973.5   588.4  5001.5  589.56  5011.5  594.72  5021.5  595.73  5041.6  595.83
  5051.6  596.37  5061.6  597.35  5071.6  599.06    5091  599.58  5101.6  601.12
  5141.7  603.55  5156.2  605.72  5161.7  606.36  5181.7  610.11  5187.9   610.5
#Mann= 4 ,-1 , 0
  4780.5     .05       0  4969.5    .033       0  4973.5     .05       0
  5156.2      .1       0
Bank Sta=4969.5,4973.5
XS Rating Curve= 0 ,0
Exp/Cntr=0.3,0.1

Type RM Length L Ch R = 1 ,17331   ,138,138,138
BEGIN DESCRIPTION:
Farris Branch 32.8
END DESCRIPTION:
XS GIS Cut Line= 3
      2400465.96      7029052.74      2400506.28      7028896.83
      2400495.53       7028649.5
#Sta/Elev= 30
  4751.7  602.78  4782.1  603.22  4787.2   602.4  4795.8  597.67  4806.2  596.35
  4816.5  595.55  4847.5  593.87  4857.8  593.95  4863.3  594.49  4868.5  593.16
  4878.5  593.44  4898.8  593.04    4904  592.33  4929.6  592.05    4965  588.92
    4970  589.56  4977.6  588.41  4977.9  587.91  4981.4  587.91  4981.6  588.41
  5029.7  588.44  5039.7  593.86  5069.7  596.87  5079.7   597.5  5089.7  599.51
  5099.7  602.24  5109.8  603.99  5129.8  605.35  5139.8  606.44  5160.3  607.64
#Mann= 3 ,-1 , 0
  4751.7     .05       0  4977.6    .033       0  4981.6     .05       0
Bank Sta=4977.6,4981.6
XS Rating Curve= 0 ,0
Exp/Cntr=0.3,0.1

Type RM Length L Ch R = 1 ,17193   ,203,203,203
BEGIN DESCRIPTION:
Farris Branch 32.0
END DESCRIPTION:
XS GIS Cut Line= 3
      2400449.82      7029122.66      2400603.06      7028904.89
      2400681.04      7028697.87
#Sta/Elev= 30
  4717.7  606.66    4754  606.23  4769.9  605.77  4776.5   604.2  4812.2  601.59
    4827  602.18  4841.9  600.13    4848  600.55  4855.5  594.95  4862.8  593.93
  4904.6  591.51  4913.3  590.75  4928.1  588.38  4953.1  588.33  4953.4  587.83
  4956.9  587.83  4957.1  588.33  4977.7  588.35  4983.9   590.5  4990.6  588.49
  4999.9  593.12  5010.1  595.16  5015.5  594.97  5040.3  597.84  5075.9  600.28
  5095.4  602.45  5117.4  603.31  5125.6  604.43  5149.5  605.88  5205.2  608.11
#Mann= 4 ,-1 , 0
  4717.7    .075       0    4754     .05       0  4953.1    .033       0
  4957.1     .05       0
Bank Sta=4953.1,4957.1
XS Rating Curve= 0 ,0
Exp/Cntr=0.3,0.1

Type RM Length L Ch R = 1 ,16990   ,238,238,238
BEGIN DESCRIPTION:
Farris Branch 31.0
END DESCRIPTION:
XS GIS Cut Line= 3
      2400648.75      7029206.01      2400810.07      7028937.15
      2400793.99        7028755.
#Sta/Elev= 30
  4761.3  600.49  4803.3  600.78  4846.7  597.87  4917.3  594.68  4926.4  594.07
  4932.2  594.44  4954.9  594.04  4963.3  589.02  4969.1   587.1  4978.2  574.76
  4982.7  574.11  4982.9  573.61  4986.4  573.61  4986.7  574.11  4990.5  575.81
  5000.2  578.58  5013.2  586.61  5021.6  589.92  5027.4  588.69    5043  591.64
  5048.8  591.18  5058.5  592.43  5064.4  591.98  5070.3  592.85  5122.2  596.24
  5140.5  597.02  5152.3  598.24  5232.6   600.4  5252.6  601.23  5257.7  602.03
#Mann= 4 ,-1 , 0
  4761.3      .1       0  4917.3     .05       0  4982.7     .05       0
  4986.7     .05       0
Bank Sta=4982.7,4986.7
XS Rating Curve= 0 ,0
Exp/Cntr=0.3,0.1

Type RM Length L Ch R = 1 ,16752   ,221,221,221
BEGIN DESCRIPTION:
Farris Branch 30.6
END DESCRIPTION:
XS GIS Cut Line= 3
       2400632.6      7029283.95      2400799.31      7029278.57
       2401104.9      7028836.27
#Sta/Elev= 30
  4654.6  605.44    4681   601.5  4792.2  600.61  4818.7  594.28  4827.7  594.56
  4833.8  591.23  4842.6  591.47  4848.6  590.09  4863.5  590.96  4920.3  589.13
  4935.2  585.42  4941.2  579.99    4950  576.23  4954.1   572.4  4954.4   571.9
  4958.1   572.4  4985.9  572.96  4991.9  576.26  5000.7  577.52  5006.8  582.94
  5021.7  586.14  5027.8  588.83  5036.6  589.44  5042.6   591.7  5050.6  591.08
  5057.5  592.43  5063.6  595.49  5123.1  597.98  5302.2  599.66    5359  602.87
#Mann= 4 ,-1 , 0
  4654.6      .1       0  4792.2     .05       0  4954.1     .05       0
  4958.1     .05       0
Bank Sta=4954.1,4958.1
XS Rating Curve= 0 ,0
Exp/Cntr=0.3,0.1

Type RM Length L Ch R = 1 ,16531   ,206,206,206
BEGIN DESCRIPTION:
Farris Branch 30.4
END DESCRIPTION:
XS GIS Cut Line= 3
      2400664.86      7029318.89      2400928.35      7029372.66
      2401234.44      7028929.65
#Sta/Elev= 30
  4685.5  602.27    4763  600.16  4791.8  598.11  4832.6  589.18  4904.1  587.95
  4912.6  584.71    4943  582.24    4948  580.67  4952.2  578.87  4961.6  579.42
  4970.1  578.48  4978.9  580.84  4999.9  572.39  5018.8   570.4  5019.1   569.9
  5022.8   570.4  5050.6  573.74  5056.7  576.42  5086.4   579.1  5107.4  584.42
  5122.2  584.98  5143.2  590.68  5244.6  595.69  5310.1  595.52    5352  600.37
  5395.2  600.63  5408.8  602.55  5459.5  602.27  5474.4  605.66  5492.9  605.78
#Mann= 7 ,-1 , 0
  4685.5      .1       0    4763     .05       0    4943    .075       0
    4948     .12       0  4961.6     .05       0  5018.8     .05       0
  5022.8     .05       0
Bank Sta=5018.8,5022.8
XS Rating Curve= 0 ,0
Exp/Cntr=0.3,0.1

Type RM Length L Ch R = 1 ,16325   ,223,223,223
BEGIN DESCRIPTION:
Farris Branch 30.0
END DESCRIPTION:
XS GIS Cut Line= 3
      2400557.39      7029437.19      2400982.12      7029515.15
       2401304.4      7029410.41
#Sta/Elev= 30
  4660.6  605.94  4692.7  606.15  4700.8  599.85    4799  598.88  4870.3  596.28
  4885.9  591.28  4906.2  589.96  4946.9  589.71  4957.1  580.24  4967.2  578.94
  4981.7  573.13  4987.6  569.18  4995.7  568.01    4996  567.51  4999.7  568.01
  5007.9  574.47    5028  575.65  5034.8  581.66  5039.9   580.8  5048.6  583.03
  5068.9  583.96  5087.9  581.91  5125.6  582.25  5131.2  585.88  5141.7  588.62
  5183.8  592.73  5194.8  596.35  5253.4  599.45  5397.8  612.01  5431.3  613.86
#Mann= 6 ,-1 , 0
  4660.6      .1       0    4799    .075       0  4995.7     .07       0
  4999.7    .075       0    5028     .12       0  5397.8     .05       0
Bank Sta=4995.7,4999.7
XS Rating Curve= 0 ,0
Exp/Cntr=0.3,0.1

Type RM Length L Ch R = 1 ,16102   ,412,412,412
BEGIN DESCRIPTION:
Farris Branch 29.0
END DESCRIPTION:
XS GIS Cut Line= 3
      2400654.16      7029775.91      2400893.41      7029722.15
      2401284.93      7029550.52
#Sta/Elev= 30
  4713.2  600.96  4763.6  599.74  4779.7  597.83  4820.7  595.97  4841.1  592.89
  4892.4   592.3  4898.7  589.46  4980.3  583.35  4996.5  581.32  5001.9   578.1
  5008.2  568.03  5017.1  565.58  5017.4  565.08  5021.1  565.58  5040.9  573.07
    5072  573.97  5077.5  577.33  5084.6  577.95  5100.9  577.47  5106.5  575.66
  5139.2  576.42  5147.6  577.91  5153.1  583.35  5176.5  585.82  5228.7  594.47
  5313.9  603.32  5322.1  605.18  5357.6  606.39  5379.8  608.27  5385.9   609.9
#Mann= 4 ,-1 , 0
  4713.2    .075       0  4980.3     .12       0  5017.1     .07       0
  5021.1     .12       0
Bank Sta=5017.1,5021.1
XS Rating Curve= 0 ,0
Exp/Cntr=0.3,0.1

Type RM Length L Ch R = 1 ,15690   ,327,327,327
BEGIN DESCRIPTION:
Farris Branch 28.0
END DESCRIPTION:
XS GIS Cut Line= 4
      2400686.41      7029888.83      2401025.13      7029910.33
      2401185.67      7029987.21      2401431.12      7029961.41
#Sta/Elev= 30
  4582.6  599.47  4649.2  596.08  4675.2  592.68  4726.8  591.51  4745.5  587.11
  4785.6  584.91  4805.6  581.34  4875.8  580.02  4885.8  577.08  4915.9     563
    4955  563.79  4960.5   563.1  4977.6  568.26  4983.2  566.26  5000.3  564.06
  5003.9  562.05  5004.1  561.55  5007.9  562.05    5023  563.15  5028.5  569.13
  5051.2  575.86  5104.2  582.67  5119.8  587.83  5124.8  587.04  5133.5  589.85
  5153.6  592.32  5229.9  598.35  5274.3  600.77  5304.4  603.99  5346.8   604.9
#Mann= 6 ,-1 , 0
  4582.6    .075       0  4649.2     .05       0  4726.8     .12       0
  5003.9     .07       0  5007.9     .12       0  5229.9     .05       0
Bank Sta=5003.9,5007.9
XS Rating Curve= 0 ,0
Exp/Cntr=0.3,0.1

Type RM Length L Ch R = 1 ,15363   ,371,371,371
BEGIN DESCRIPTION:
Farris Branch 27.0
END DESCRIPTION:
XS GIS Cut Line= 3
      2400799.31       7030195.3        2401129.        7030210.
      2401344.47      7030224.83
#Sta/Elev= 30
  4677.1  588.34  4706.8  588.16  4716.8  586.55  4746.9  584.53  4816.9   584.2
  4826.9  583.62  4836.9  581.62    4847   578.2    4867  578.22  4878.2  576.92
    4907  576.48    4927   577.4    4937  576.12  4947.1   574.1  4987.1  562.74
  4997.1  561.05  5002.6  558.59  5002.9  558.09  5006.6  558.59  5017.1  559.01
  5037.2  566.85  5047.2  572.71  5057.2  579.93  5067.3  584.29  5076.1  586.13
  5119.8  590.48  5167.5  594.69  5177.5  597.53  5187.5  599.01  5223.1  599.76
#Mann= 5 ,-1 , 0
  4677.1     .05       0  4878.2     .12       0  5002.6     .07       0
  5006.6     .12       0  5119.8     .05       0
Bank Sta=5002.6,5006.6
XS Rating Curve= 0 ,0
Exp/Cntr=0.3,0.1

Type RM Length L Ch R = 1 ,14992   ,348,348,348
BEGIN DESCRIPTION:
Farris Branch 26.0
END DESCRIPTION:
XS GIS Cut Line= 3
      2400721.37      7030418.44        2400979.        7030510.
      2401242.92      7030579.74
#Sta/Elev= 30
  4731.1  586.03  4747.6  585.44  4760.4  581.51    4771  580.02  4809.3  579.79
  4927.4  574.85  4940.8  574.65  4951.5  575.99  4972.7  569.59  4983.3  563.45
  4994.4  559.46  4999.9  555.52  5000.1  555.02  5003.9  555.52  5007.1  555.52
  5018.5  562.72  5027.2  570.52  5062.3  577.46  5097.4  577.87  5102.6  580.68
  5118.3  579.61  5128.6  581.24  5137.7   584.8  5149.3  586.32  5159.7  586.54
  5211.4  585.87  5218.2  592.59  5223.4     592  5232.1  593.62  5277.5  593.25
#Mann= 5 ,-1 , 0
  4731.1     .05       0  4999.9     .05       0  5003.9     .05       0
  5018.5     .12       0  5159.7     .05       0
Bank Sta=4999.9,5003.9
XS Rating Curve= 0 ,0
Exp/Cntr=0.3,0.1

Type RM Length L Ch R = 1 ,14644   ,384,384,384
BEGIN DESCRIPTION:
Farris Branch 25.0
END DESCRIPTION:
XS GIS Cut Line= 4
      2400632.63       7030886.2      2400865.74      7030841.63
      2401003.63      7030765.23      2401199.89      7030708.77
#Sta/Elev= 30
  4692.9  591.73    4791  583.33    4801  579.96    4903  577.51  4910.2   575.9
  4929.3  566.68  4941.8  566.99  4952.8  563.73  4956.8  563.16  4967.3   553.6
  4967.5   553.1  4971.3   553.6  4979.6  553.87  4991.1  559.92  5001.3  561.15
    5014  567.33  5028.8  569.12  5036.9  567.94  5050.5  571.21  5066.6  571.14
  5072.3  573.44  5087.9   573.8  5103.9  579.55  5161.1   579.2  5166.3  582.73
  5173.3  583.13    5186   586.2  5239.1  587.24    5260  592.24  5292.1   592.7
#Mann= 6 ,-1 , 0
  4692.9     .05       0  4952.8     .12       0  4967.3     .07       0
  4971.3     .12       0  5173.3     .05       0    5186     .12       0
Bank Sta=4967.3,4971.3
XS Rating Curve= 0 ,0
Exp/Cntr=0.3,0.1

Type RM Length L Ch R = 1 ,14260   ,352,352,352
BEGIN DESCRIPTION:
Farris Branch 24.0
END DESCRIPTION:
XS GIS Cut Line= 3
      2400694.47      7031157.73      2401014.38      7031155.04
      2401494.79      7031050.37
#Sta/Elev= 30
    4769   591.3  4803.5  589.12  4813.5  585.04  4853.5  584.02  4873.5  580.69
  4903.5  581.04  4933.5  579.18  4953.5  571.93  4963.5  570.06  5006.7  565.64
  5023.5  558.14  5063.5  553.89  5071.5  551.66  5071.8  551.16  5075.5  551.66
  5083.5  552.72  5103.9  564.39  5114.1  567.11  5151.8  567.33  5257.4  569.33
    5280  571.84  5298.3  579.56  5308.6  581.54  5349.5  581.25  5380.2  585.96
  5422.1  586.71  5441.6  591.66    5503  592.63  5523.5  596.09  5580.6  597.55
#Mann= 5 ,-1 , 0
    4769     .05       0  5006.7     .12       0  5071.5     .05       0
  5075.5     .12       0  5151.8     .05       0
Bank Sta=5071.5,5075.5
XS Rating Curve= 0 ,0
Exp/Cntr=0.3,0.1

Type RM Length L Ch R = 1 ,13908   ,342,342,342
BEGIN DESCRIPTION:
Farris Branch 23.0
END DESCRIPTION:
XS GIS Cut Line= 3
       2400823.5       7031488.4        2401129.        7031310.
      2401280.55       7031230.3
#Sta/Elev= 30
  4645.7  585.15  4708.1   582.7  4713.8  583.28  4729.5  580.56  4735.3  580.72
  4756.8  577.74  4779.4  572.88  4809.7  569.23  4831.2  568.67  4846.9  567.05
  4905.6  565.56  4918.4  563.44  4932.9  558.03    4957  555.77  4964.3  556.18
  4970.1  554.16  5002.3  553.54  5013.3  550.24  5020.1  549.99  5020.3  549.49
  5024.1  549.99  5029.7  550.92  5035.4  559.31  5044.7  564.75  5095.8   575.2
  5101.5  578.67  5112.2  576.62  5117.9  579.02  5123.8  579.37  5170.7  579.22
#Mann= 5 ,-1 , 0
  4645.7     .05       0  4831.2     .12       0    4957     .05       0
  5020.1    .033       0  5024.1     .05       0
Bank Sta=5020.1,5024.1
XS Rating Curve= 0 ,0
Exp/Cntr=0.3,0.1

Type RM Length L Ch R = 1 ,13566   ,373,373,373
BEGIN DESCRIPTION:
Farris Branch 22.0
END DESCRIPTION:
XS GIS Cut Line= 4
      2400909.54      7031706.14      2401077.37      7031621.06
      2401189.12      7031483.02      2401429.04      7031359.98
#Sta/Elev= 30
  4768.3  584.73  4823.7  579.55  4915.3   573.4  4944.6  569.79  4965.6  569.75
  4972.1  566.16    4980  554.64  4986.4  549.29  4992.4  546.36  4992.6  545.86
  4996.4  546.36  5008.8  547.71  5022.2  552.38  5029.6  553.35  5050.4  552.73
  5079.2  554.01  5093.5  557.64    5100  561.08  5107.9  562.71  5122.3  563.26
  5128.7  562.06    5179  564.52  5234.4  570.93  5262.2  576.14  5278.8  576.08
  5313.7     579  5345.4  584.64  5395.4  586.21  5400.8  591.79  5403.7  591.79
#Mann= 4 ,-1 , 0
  4768.3     .05       0  4915.3     .12       0  4992.4     .07       0
  4996.4     .12       0
Bank Sta=4992.4,4996.4
XS Rating Curve= 0 ,0
Exp/Cntr=0.3,0.1

Type RM Length L Ch R = 1 ,13193   ,464,464,464
BEGIN DESCRIPTION:
Farris Branch 21.0
END DESCRIPTION:
XS GIS Cut Line= 3
       2401014.4      7031749.16        2401329.        7031760.
       2401568.2       7031762.6
#Sta/Elev= 30
  4685.2  578.29  4716.4  576.86  4759.8   573.3  4779.9  572.55  4809.9  569.59
  4829.9  568.52  4839.9  567.25  4849.8  566.63  4854.8  566.96  4879.9  563.95
  4919.9  561.68    4950  561.18    4960  559.04    4970  552.99    4988  543.84
  4988.2  543.34  4991.7  543.34    4992  543.84  5002.5  543.89    5010  554.19
    5020   563.3    5030  564.32    5040  564.57    5060  566.74    5090  567.77
    5120  571.04    5180   573.7    5210  578.11    5230  582.04  5239.2  582.99
#Mann= 4 ,-1 , 0
  4685.2     .05       0  4716.4     .12       0    4988     .07       0
    4992     .12       0
Bank Sta=4988,4992
XS Rating Curve= 0 ,0
Exp/Cntr=0.3,0.1

Type RM Length L Ch R = 1 ,12729   ,436,436,436
BEGIN DESCRIPTION:
Farris Branch 20.0
END DESCRIPTION:
XS GIS Cut Line= 3
      2401000.98      7032157.79      2401216.01      7032171.23
      2401549.32      7032165.86
#Sta/Elev= 30
  4719.9  580.83  4727.9  580.37    4738   576.6    4748  571.74    4758  572.53
  4782.9   571.4  4798.1  569.29  4818.1  567.64  4834.3  565.09  4868.2  561.71
  4908.3  560.01  4934.3  556.77  4948.3  556.99  4958.3   556.1  4968.3  556.62
  4988.3  555.21  5008.3   545.6  5026.4  540.27  5026.6  539.77  5030.1  539.77
  5030.4  540.27  5048.4  551.67  5058.4  553.46  5068.4  553.26  5078.4  554.47
  5088.4  556.29  5098.4  560.75  5128.4  561.79  5218.4  569.41  5268.7  572.12
#Mann= 4 ,-1 , 0
  4719.9     .05       0  4782.9     .12       0  5026.4     .07       0
  5030.4     .12       0
Bank Sta=5026.4,5030.4
XS Rating Curve= 0 ,0
Exp/Cntr=0.3,0.1

Type RM Length L Ch R = 1 ,12293   ,215,215,215
BEGIN DESCRIPTION:
Farris Branch 19.0
END DESCRIPTION:
XS GIS Cut Line= 3
      2401006.35      7032421.26      2401186.43      7032453.51
      2401568.15      7032305.66
#Sta/Elev= 30
  4595.9   576.2  4629.1  575.27  4639.2  572.81  4666.7  571.35  4674.3  572.02
  4710.3  570.57  4728.1  568.08  4780.9  566.27  4835.3  562.38  4845.9  562.49
  4854.5  560.94  4878.2  559.83  4914.4  559.37  4931.7  555.94    4939  556.28
  4968.9  546.95  4985.4  544.85  4993.5  542.89  4998.8     539  5015.5  538.37
  5015.8  537.87  5019.5  538.37  5023.4   544.3  5028.8  550.84    5039   555.7
  5083.3  559.96  5102.5  560.76    5114  563.17  5162.3  568.16  5188.2  568.38
#Mann= 6 ,-1 , 0
  4595.9     .05       0  4666.7     .12       0  4780.9     .05       0
  4878.2     .12       0  5015.5     .07       0  5019.5     .12       0
Bank Sta=5015.5,5019.5
XS Rating Curve= 0 ,0
Exp/Cntr=0.3,0.1

Type RM Length L Ch R = 1 ,12078   ,216,216,216
BEGIN DESCRIPTION:
Farris Branch 18.0
END DESCRIPTION:
XS GIS Cut Line= 3
      2401224.03      7032585.24       2401517.1      7032550.29
      2401576.23       7032418.6
#Sta/Elev= 30
  4743.2  572.02  4749.2  572.17  4758.3   571.5  4778.4  569.76  4798.6  567.11
  4861.8  562.55  4879.1  560.72  4889.2  560.13  4914.3  556.86  4919.4  556.85
  4949.6  547.73  4969.8   544.2  4989.9   538.7  4994.8   538.1    4995   537.6
  4998.5   537.6  4998.8   538.1  5001.8  538.21    5010  551.12  5020.1  551.71
  5030.2  550.36  5049.6  551.01  5055.1  551.57  5060.6  555.59  5083.8  556.61
  5124.7  557.15  5153.3  559.03  5176.5   563.1    5180  562.48  5182.7  562.48
#Mann= 4 ,-1 , 0
  4743.2     .05       0  4861.8     .12       0  4994.8     .07       0
  4998.8     .12       0
Bank Sta=4994.8,4998.8
XS Rating Curve= 0 ,0
Exp/Cntr=0.3,0.1

Type RM Length L Ch R = 1 ,11862   ,281,281,281
BEGIN DESCRIPTION:
Farris Branch 17.5
END DESCRIPTION:
XS GIS Cut Line= 3
      2401342.41      7032762.67       2401471.4      7032762.67
      2401871.99      7032569.09
#Sta/Elev= 30
  4751.1  566.82  4828.7  561.95  4924.1  554.14    4933  551.85  4941.1  552.41
  4946.7  548.88  4977.4  545.04  4999.6  544.09  5012.4   535.8  5012.7   535.3
  5016.4   535.8  5021.8  541.22  5031.5  548.28    5044  551.84  5104.8  556.11
  5127.4  556.71    5133  557.92    5144  557.81    5150  558.35  5155.6  560.41
  5172.6  560.04  5178.2   561.2  5217.8  562.59  5223.4  565.05  5240.4  565.56
    5246  566.71    5255   565.6    5263  565.93  5299.5  571.19    5325  573.42
#Mann= 4 ,-1 , 0
  4751.1     .05       0  4828.7     .12       0  5012.4     .07       0
  5016.4     .12       0
Bank Sta=5012.4,5016.4
XS Rating Curve= 0 ,0
Exp/Cntr=0.3,0.1

Type RM Length L Ch R = 1 ,11581   ,338,338,338
BEGIN DESCRIPTION:
Farris Branch 17.0
END DESCRIPTION:
XS GIS Cut Line= 3
      2401369.23       7032824.5      2401673.03      7032883.64
      2402094.56      7032776.25
#Sta/Elev= 30
  4580.1  565.54  4583.8  564.79  4635.5  562.56  4664.3  559.91  4712.3   556.7
    4804  552.97    4937  550.54  4957.7  547.53    4964  545.37  4969.1  539.51
  4986.6  535.61  4986.9  535.11  4990.6  535.61    4999   535.7    5010  549.75
  5019.6  551.54  5029.9  550.52  5040.2  551.68  5045.8  550.59  5050.9  554.67
  5060.9  553.88  5071.2  558.29  5086.6   560.3  5122.4  562.47  5133.1  564.34
  5215.7   571.2  5236.3  573.74  5289.5  575.56  5308.5  575.35  5324.6  573.99
#Mann= 5 ,-1 , 0
  4580.1     .05       0  4664.3     .12       0  4986.6     .07       0
  4990.6     .12       0  5289.5     .05       0
Bank Sta=4986.6,4990.6
XS Rating Curve= 0 ,0
Exp/Cntr=0.3,0.1

Type RM Length L Ch R = 1 ,11243   ,155,155,155
BEGIN DESCRIPTION:
Farris Branch 16.2
END DESCRIPTION:
XS GIS Cut Line= 4
      2401156.82      7033168.62      2401533.23      7033106.78
      2401713.35      7033044.94      2402019.86      7033012.68
#Sta/Elev= 30
  4545.6  567.25  4560.1  567.09  4570.5  564.55  4626.7  565.33  4631.8   561.2
    4688  563.11    4693  559.99  4749.2  561.77  4754.3  558.74  4810.4  560.46
  4815.5  556.24    4862  555.26  4927.1  550.75  4936.9  547.37  4954.3  543.25
  4966.7  536.46  4992.7   535.6    4998  537.62  5017.7  535.38    5024  539.29
  5027.1  535.35  5027.5  534.85  5031.5  535.35  5038.9  541.28  5117.4  545.49
  5210.6  558.19    5274  564.09  5354.4  567.67  5425.4  567.38  5425.7  567.38
#Mann= 6 ,-1 , 0
  4545.6     .05       0  4560.1    .075       0  4936.9     .05       0
  5027.1     .05       0  5031.5     .05       0  5425.4     .12       0
Bank Sta=5027.1,5031.5
XS Rating Curve= 0 ,0
Exp/Cntr=0.3,0.1

Type RM Length L Ch R = 1 ,11088   ,296,296,296
BEGIN DESCRIPTION:
Farris Branch 16.0
END DESCRIPTION:
XS GIS Cut Line= 3
      2401312.79      7033278.83      2401576.25      7033225.06
      2401915.87      7033171.58
#Sta/Elev= 30
  4622.9  569.65  4649.7  569.59  4693.8  568.43  4739.2  563.51  4744.3  564.09
  4789.8  560.88    4864  554.02  4890.6  550.65  4895.9  550.54  4924.9  545.39
  4945.2   541.3  4963.2  534.27  4963.6  533.77  4967.2  533.77  4967.6  534.27
  4975.6  535.63  4985.7  539.03  5005.9  541.01  5026.2  545.36  5046.4  547.34
  5107.2  550.97  5127.4  551.63  5137.5   553.4  5157.8  554.31    5178  560.35
  5188.1  561.61  5198.3  562.07  5213.5  561.84  5218.6  565.25  5235.6  564.57
#Mann= 3 ,-1 , 0
  4622.9    .075       0  4963.2     .07       0  4967.6    .075       0
Bank Sta=4963.2,4967.6
XS Rating Curve= 0 ,0
Exp/Cntr=0.3,0.1

Type RM Length L Ch R = 1 ,10792   ,392,392,392
BEGIN DESCRIPTION:
Farris Branch 15.0
END DESCRIPTION:
XS GIS Cut Line= 3
      2401689.13       7033520.8      2401904.22      7033383.68
      2401944.28      7033162.05
#Sta/Elev= 30
  4671.1  559.64  4695.8  557.65    4711  557.52  4736.9  557.71  4742.9  556.38
  4779.2  553.52  4809.7  552.77  4903.7  547.94  4918.9  546.05  4924.8  543.33
  4930.6   542.8  4950.2  537.72  4960.4  533.97  4968.4  533.11  4968.8  532.61
  4972.8  533.11  4978.4  537.61  4990.9  538.51    5001  538.09  5011.2  540.85
  5031.5   547.5    5037   551.6  5042.1   550.7  5072.2  554.63  5101.5  555.77
  5112.8  557.14    5123  556.93  5143.3   563.1  5149.1  565.93  5151.4  565.47
#Mann= 6 ,-1 , 0
  4671.1     .12       0  4695.8     .05       0    4711     .12       0
  4968.4     .07       0  4972.8     .12       0  5101.5     .05       0
Bank Sta=4968.4,4972.8
XS Rating Curve= 0 ,0
Exp/Cntr=0.3,0.1

Type RM Length L Ch R = 1 ,10400   ,103,103,103
BEGIN DESCRIPTION:
Farris Branch 14.5
END DESCRIPTION:
XS GIS Cut Line= 3
      2401968.76      7033641.75      2402251.02      7033544.98
      2402307.28      7033113.62
#Sta/Elev= 30
  4616.1  555.98  4697.1  553.59  4722.1   551.7  4753.8  548.21  4790.9  546.56
  4859.5  545.46  4870.1  544.38  4914.5  543.39  4949.8   543.6  4959.8  541.26
  4969.9  536.89    4980  536.14  4990.1  536.57  5000.2  535.58  5015.1  532.88
  5018.2  530.93  5018.6  530.43  5022.6  530.93  5040.5  539.22  5050.6  541.79
  5070.8   546.7  5080.9   547.2    5101  550.44  5151.5  553.64  5181.7  556.76
  5232.1  557.96  5262.4   560.2  5282.6  560.44  5340.6  563.99  5349.5   564.8
#Mann= 4 ,-1 , 0
  4616.1     .12       0  5018.2     .07       0  5022.6     .12       0
  5340.6    .075       0
Bank Sta=5018.2,5022.6
XS Rating Curve= 0 ,0
Exp/Cntr=0.3,0.1

Type RM Length L Ch R = 1 ,10297   ,356,356,356
BEGIN DESCRIPTION:
Farris Branch 14.0
END DESCRIPTION:
XS GIS Cut Line= 3
      2402285.96      7033937.49      2402366.62      7033644.45
      2402361.24      7033195.52
#Sta/Elev= 30
  4511.6  561.33  4571.2  558.31    4578  555.53  4623.1  555.34  4643.8  553.92
  4664.6  550.87  4696.7     550  4706.1  548.38  4731.1  547.63  4744.1  546.06
  4778.7  543.76  4815.3  536.39    4840  534.66  4846.9  535.54    4870  543.03
    4960  541.69    4970  539.59    4980  533.24  4987.8  530.62  4988.2  530.12
  4992.2  530.62    5000  530.71    5020  540.87  5029.6  544.33  5034.6  543.44
    5040  545.32    5090  548.56    5170  557.35    5220  559.73  5264.5  560.09
#Mann= 5 ,-1 , 0
  4511.6     .12       0  4744.1     .05       0  4846.9     .12       0
  4987.8     .07       0  4992.2     .12       0
Bank Sta=4987.8,4992.2
XS Rating Curve= 0 ,0
Exp/Cntr=0.3,0.1

Type RM Length L Ch R = 1 ,9941    ,477,477,477
BEGIN DESCRIPTION:
Farris Branch 13.0
END DESCRIPTION:
XS GIS Cut Line= 3
       2402694.6      7033918.65      2402697.29      7033593.37
      2402595.12      7033117.51
#Sta/Elev= 30
  4638.9  560.77  4657.6  557.92  4707.6  554.24  4747.6  549.64  4767.6  553.84
  4777.6  553.87  4787.6  553.55  4807.6   549.4  4815.1  549.78  4827.6  549.32
  4837.6  550.72  4857.6  549.32  4917.6  543.07  4936.2  537.97  4947.6  535.29
  4957.6  530.78  4973.9   530.1  4974.5   529.6  4978.7   530.1  4988.1  530.57
  5018.8  537.27  5025.7   540.2  5049.5  541.17  5124.5  541.29  5218.1  543.93
  5274.5  546.69  5316.9  549.85  5335.8  550.17  5417.7  557.63  5450.9  558.03
#Mann= 5 ,-1 , 0
  4638.9     .12       0  4815.1     .05       0  4936.2     .12       0
  4973.9     .07       0  4978.7     .12       0
Bank Sta=4973.9,4978.7
XS Rating Curve= 0 ,0
Exp/Cntr=0.3,0.1

Type RM Length L Ch R = 1 ,9464    ,507,507,507
BEGIN DESCRIPTION:
Farris Branch 12.0
END DESCRIPTION:
XS GIS Cut Line= 3
      2403069.69      7033895.27      2403099.78      7033639.51
      2402889.17      7032987.62
#Sta/Elev= 30
  4582.5  558.85  4597.9  557.59  4621.2  553.94  4651.8  554.36  4668.4  553.66
  4704.3  548.47  4748.9  546.18  4792.4  542.16  4819.4  542.03  4902.6  538.97
  4921.1  537.27  4934.1  534.75  4953.1  533.67  4965.6   531.4  4985.2  531.35
  4996.3  529.77  5014.7  527.77  5015.3  527.27  5019.6  527.77  5022.4  531.24
  5028.7  533.25  5074.7  533.81  5086.5  534.37  5102.2  539.42  5219.9  543.54
  5278.7  546.74  5291.4  548.53  5301.9  548.36    5386  553.24  5525.1     554
#Mann= 6 ,-1 , 0
  4582.5     .05       0  4651.8     .12       0  4996.3     .05       0
  5014.7    .033       0  5019.6     .05       0  5074.7     .12       0
Bank Sta=5014.7,5019.6
XS Rating Curve= 0 ,0
Exp/Cntr=0.3,0.1

Type RM Length L Ch R = 1 ,8957    ,434,434,434
BEGIN DESCRIPTION:
Farris Branch 11.0
END DESCRIPTION:
XS GIS Cut Line= 3
      2403094.73      7033915.35      2403460.83      7033514.14
      2403731.61      7032817.12
#Sta/Elev= 30
  4345.4  556.22  4387.7  555.61  4401.8  554.43  4408.6  555.25  4443.5  551.88
  4515.1  548.45  4564.7  543.53  4642.4  538.45    4770  535.75  4805.5  536.01
  4854.5   534.7  4897.8  535.69  4927.7  532.25  4968.1  531.91  4982.1  530.69
  4987.3  525.26  5036.6  529.97  5061.1   532.9  5075.4  532.73  5085.7  535.81
    5091  533.77  5096.8  538.18  5107.5  540.77  5115.6  545.28  5139.7  545.64
  5145.5   547.9  5199.7  551.21  5308.8  557.18    5483  559.07  5636.3  565.37
#Mann= 6 ,-1 , 0
  4345.4     .05       0  4443.5     .12       0  4805.5     .05       0
  4982.1    .033       0  5036.6     .05       0  5199.7     .12       0
Bank Sta=4982.1,5036.6
XS Rating Curve= 0 ,0
Exp/Cntr=0.3,0.1

Type RM Length L Ch R = 1 ,8523    ,411,411,411
BEGIN DESCRIPTION:
Farris Branch 10.0
END DESCRIPTION:
XS GIS Cut Line= 3
      2403144.89      7034060.75      2403601.24      7033654.55
      2404071.15      7033524.58
#Sta/Elev= 30
  4308.5  557.79  4354.2  555.53  4368.3  555.33  4375.8  556.52    4390  556.24
  4410.9  554.07  4467.8  553.19  4517.1  551.45  4548.8  547.62  4609.1  542.16
  4630.8  541.24    4645  539.29  4708.6  537.07  4738.6  535.16  4757.9  535.65
  4765.4  534.47  4779.6  533.86  4843.2  532.61  4878.3  533.64  4885.8  532.91
  4977.1  530.64  5186.9  534.83  5207.6  540.91  5215.3  544.39  5220.5  543.13
  5228.4  545.76  5280.3  549.41  5311.4  553.06  5373.6  555.26    5407  555.36
#Mann= 5 ,-1 , 0
  4308.5     .05       0  4548.8     .12       0  4738.6     .05       0
  4878.3    .033       0  5186.9     .05       0
Bank Sta=4878.3,5186.9
XS Rating Curve= 0 ,0
Exp/Cntr=0.3,0.1

Type RM Length L Ch R = 1 ,8112    ,407,407,407
BEGIN DESCRIPTION:
Farris Branch 9.0
END DESCRIPTION:
XS GIS Cut Line= 3
       2403144.9      7034366.63        2403779.        7034010.
      2404029.04      7033859.98
#Sta/Elev= 30
  4277.1  557.01  4445.9  552.75  4483.5  554.09  4505.2  552.74  4521.1  555.07
  4526.8  553.66  4531.9  554.31  4542.8  556.41  4548.5  555.19  4564.5  556.79
  4580.1  556.31  4607.8  551.86  4637.5  554.16  4675.8  553.05  4688.8  552.81
  4704.7   549.7  4710.4     551  4726.4   547.5  4732.1  549.31    4748  545.78
  4753.8  547.77  4769.7  544.51  4775.4  545.95  4791.4  543.59  4798.1  539.63
    4821     535  5060.7  530.62  5113.5  534.04    5129  536.82  5296.2  550.34
#Mann= 5 ,-1 , 0
  4277.1     .05       0  4531.9     .12       0  4675.8     .05       0
    4821    .033       0  5113.5     .05       0
Bank Sta=4821,5113.5
XS Rating Curve= 0 ,0
Exp/Cntr=0.3,0.1
