--- Golf Course Creek Tr 1.prj (project) ---

Proj Title=Golf Course Creek Tr 1 Base Level Engineering
Current Plan=p01
Default Exp/Contr=0.3,0.1
English Units
Geom File=g01
Flow File=f01
Plan File=p01
Y Axis Title=Elevation
X Axis Title(PF)=Main Channel Distance
X Axis Title(XS)=Station
BEGIN DESCRIPTION:
Golf Course Creek Tr 1
END DESCRIPTION:
DSS Export Rating Curves= 0
DSS Export Rating Curve Sorted= 0
DSS Export Volume Flow Curves= 0
DXF OffsetX= 0
DXF OffsetY= 0
DXF ScaleX= 1
DXF ScaleY= 10

--- Golf Course Creek Tr 1.p01 (plan) ---

Plan Title=Multiple Run
Program Version=4.10
Short Identifier=Multiple
Geom File=g01
Flow File=f01
Subcritical Flow
K Sum by GR= 0
Std Step Tol= 0.01
Critical Tol= 0.01
Num of Std Step Trials= 20
Max Error Tol= 0.3
Flow Tol Ratio= 0.001
Split Flow NTrial= 30
Split Flow Tol= 0.02
Split Flow Ratio= 0.02
Log Output Level= 0
Friction Slope Method= 1
Unsteady Friction Slope Method= 2
Unsteady Bridges Friction Slope Method= 1
Parabolic Critical Depth
Global Vel Dist= 1 , 1 , 1
Global Log Level= 0
CheckData=True
Encroach Param=-1 ,0,0, 0
BEGIN DESCRIPTION:
Multiple Run
END DESCRIPTION:
Computation Interval=1HOUR
Output Interval=1HOUR
Run HTab= 0
Run UNet= 0
Run PostProcess= 0
Run WQNet= 0
UNET Theta= 1
UNET Theta Warmup= 1
UNET ZTol= 0.02
UNET ZSATol= 0.05
UNET MxIter= 20
UNET MaxInSteps= 0
UNET DtIC= 0
UNET DtMin= 0
UNET MaxCRTS= 20
UNET WFStab= 2
UNET SFStab= 1
UNET WFX= 1
UNET SFX= 1
UNET DSS MLevel= 4
UNET DZMax Abort= 100
UNET Convert EG Bridges= 0
UNET Use Existing IB Tables=-1
UNET Froude Reduction=False
UNET Froude Limit= 1
UNET Froude Power= 10
UNET Time Slicing=0,0, 5
UNET Junction Losses=0
Instantaneous Interval=1HOUR
Write IC File= 0
Write IC File at Sim End=0
Echo Input=False
Echo Parameters=False
Echo Output=False
Write Detailed= 0
WQ AD Non Conservative
WQ ULTIMATE=-1
WQ Max Comp Step=1HOUR
WQ Output Interval=15MIN
WQ Output Selected Increments= 0
WQ Output face flow=0
WQ Output face velocity=0
WQ Output face area=0
WQ Output face dispersion=0
WQ Output cell volume=0
WQ Output cell surface area=0
WQ Output cell continuity=0
WQ Output cumulative cell continuity=0
WQ Output face conc=0
WQ Output face dconc_dx=0
WQ Output face courant=0
WQ Output face peclet=0
WQ Output face adv mass=0
WQ Output face disp mass=0
WQ Output cell mass=0
WQ Output cell source sink temp=0
WQ Output cell source sink nsm=0
WQ Output MaxMinRange=-1
WQ Daily Max Min Mean=-1
WQ Daily Range=0
WQ Daily Time=0
WQ Create Restart=0
WQ Fixed Restart=0
WQ System Summary=0
WQ Use Fixed Temperature=0
Sorting and Armoring Iterations= 10
XS Update Threshold= 0.02
Hydraulics Update Threshold= 0.02
Energy Slope Method= 1
Volume Change Method= 0
XS Weighting Method= 0
Number of US Weighted Cross Sections= 1
Number of DS Weighted Cross Sections= 1
Upstream XS Weight=0.25
Main XS Weight=0.5
Downstream XS Weight=0.25
Number of DS XS's Weighted with US Boundary= 1
Upstream Boundary Weight= 1
Weight of XSs Associated with US Boundary= 0
Number of US XS's Weighted with DS Boundary= 1
Downstream Boundary Weight= 0.5
Weight of XSs Associated with DS Boundary= 0.5
Sediment Output Level= 4
Mass or Volume Output= 0
Output Increment Type= 1
Profile and TS Output Increment= 10
XS Output Flag= 0
XS Output Increment= 10
Disregard all LS=0
Disregard all Conn=0
Disregard all Breaches=0
Disregard all Pumps=0

--- Golf Course Creek Tr 1.f01 (steady flow) ---

Flow Title=Multiple
Number of Profiles=7
Profile Names=10-year,25-year,50-year,1pct_min,100-year,1pct_plu,500-year
River Rch & RM= Golf Course Cree,Reach-1,14301
     487     651     784     468     934    1863    1324
River Rch & RM= Golf Course Cree,Reach-1,10336
     803    1108    1361     829    1653    3299    2438
River Rch & RM= Golf Course Cree,Reach-1,4800
    1083    1523    1893    1165    2325    4640    3508
Boundary for River Rch & Prof#=Golf Course Cree,Reach-1,1
Up Type=0
Dn Type=3
Dn Slope=0.005
Boundary for River Rch & Prof#=Golf Course Cree,Reach-1,2
Up Type=0
Dn Type=3
Dn Slope=0.005
Boundary for River Rch & Prof#=Golf Course Cree,Reach-1,3
Up Type=0
Dn Type=3
Dn Slope=0.005
Boundary for River Rch & Prof#=Golf Course Cree,Reach-1,4
Up Type=0
Dn Type=3
Dn Slope=0.005
Boundary for River Rch & Prof#=Golf Course Cree,Reach-1,5
Up Type=0
Dn Type=3
Dn Slope=0.005
Boundary for River Rch & Prof#=Golf Course Cree,Reach-1,6
Up Type=0
Dn Type=3
Dn Slope=0.005
Boundary for River Rch & Prof#=Golf Course Cree,Reach-1,7
Up Type=0
Dn Type=3
Dn Slope=0.005

--- Golf Course Creek Tr 1.g01 (geometry) ---

Geom Title=Existing Conditions
Program Version=4.10

River Reach=Golf Course Cree,Reach-1
Reach XY= 30
        2367529.        7039760.      2367775.94      7039868.28
      2367782.75      7040108.45      2368073.48      7040457.56
      2368232.75      7041008.45      2368425.47      7041261.47
      2368328.96      7041529.98      2368382.84      7042001.38
      2368622.94      7042251.86       2368981.3      7042365.83
      2369202.81      7042583.15      2369573.38      7042965.62
      2369925.24      7043561.56      2369982.55      7043908.53
      2370326.73      7044615.94      2370330.19       7045049.5
      2370526.76      7045365.93      2370581.07      7045904.13
      2370975.26      7046511.52      2371034.42      7046862.67
      2371384.62      7047304.38      2371912.35      7047593.33
      2372477.38      7048466.03      2372275.46      7050258.54
      2372032.09      7050518.31      2371962.55      7050827.14
       2371731.9      7050867.91      2371723.59      7051204.82
      2371561.86      7051226.28        2371329.        7051560.

Type RM Length L Ch R = 1 ,14301   ,231,231,231
BEGIN DESCRIPTION:
Golf Course Creek Tr 1 40.0
END DESCRIPTION:
XS GIS Cut Line= 3
      2367578.99      7040560.01        2367879.        7040260.
        2368479.        7039760.
#Sta/Elev= 30
  4580.8  689.51  4679.8   684.2  4722.2  684.42  4750.5  683.83  4764.7  682.87
  4792.9  682.67  4807.1   681.7  4827.4  681.73  4835.4   681.7  4906.1  677.14
  4927.6  676.49  5059.7  675.29    5060  674.79  5063.5  674.79  5063.7  675.29
  5090.3  676.16  5096.8  675.72  5189.3  676.29  5246.5  677.72  5253.1  678.95
  5275.2  679.62  5281.7  678.79  5289.5  678.87  5374.1  682.09  5445.7  685.53
    5516  690.97  5715.2  701.27  5721.7  703.09  5750.3  704.02  5786.1   706.2
#Mann= 5 ,-1 , 0
  4580.8     .05       0  4827.4     .12       0  4927.6     .05       0
  5059.7    .033       0  5063.7     .05       0
Bank Sta=5059.7,5063.7
XS Rating Curve= 0 ,0
Exp/Cntr=0.3,0.1

Type RM Length L Ch R = 1 ,14070   ,236,236,236
BEGIN DESCRIPTION:
Golf Course Creek Tr 1 39.0
END DESCRIPTION:
XS GIS Cut Line= 3
      2367779.01      7040659.99        2368029.        7040410.
      2368520.44      7040245.14
#Sta/Elev= 30
  4645.9  689.85  4649.4  689.85    4660  686.43  4674.2  684.72  4702.5  684.04
    4759  681.09  4829.7  678.44  4900.4  677.64  4914.6  676.33  4942.9   675.1
    4957  673.51  4969.2  672.89  4969.4  672.39  4972.9  672.39  4973.2  672.89
  4995.9  674.48  5052.2  674.47  5109.8  675.52  5199.2  678.13    5236  680.24
  5262.3  682.44  5293.8  683.96  5393.7  687.45    5420  689.09  5425.3   688.2
  5451.5  690.81  5456.8  690.62  5483.1  692.58  5488.3  692.33  5517.8  694.23
#Mann= 3 ,-1 , 0
  4645.9     .05       0  4969.2    .033       0  4973.2     .05       0
Bank Sta=4969.2,4973.2
XS Rating Curve= 0 ,0
Exp/Cntr=0.3,0.1

Type RM Length L Ch R = 1 ,13834   ,236,236,236
BEGIN DESCRIPTION:
Golf Course Creek Tr 1 38.0
END DESCRIPTION:
XS GIS Cut Line= 3
      2367938.85      7040717.23        2368129.        7040610.
       2368260.2      7040530.52
#Sta/Elev= 30
  4786.3  680.97  4820.9  681.73  4834.8  681.46  4856.9  680.17  4915.7  677.86
  4924.2  677.08  4931.7  675.89  4937.4  675.47  4947.2  673.86  4953.3  671.76
  4959.1  671.81  4969.2  670.22    4975  670.17  4981.6  669.36  5016.4  668.39
  5019.9  668.39  5020.2  668.89  5027.8  670.79  5033.7  670.79  5039.7  672.68
  5049.2  674.16    5055  674.19  5067.8  676.02    5086  677.02  5091.9  677.01
  5098.1  678.01  5107.4  679.07  5113.2   679.3  5128.7  681.23    5158  682.09
#Mann= 5 ,-1 , 0
  4786.3     .05       0  4856.9    .075       0  4981.6    .033       0
  5020.2    .075       0  5067.8     .05       0
Bank Sta=4981.6,5020.2
XS Rating Curve= 0 ,0
Exp/Cntr=0.3,0.1

Type RM Length L Ch R = 1 ,13598   ,70,70,70
BEGIN DESCRIPTION:
Golf Course Creek Tr 1 37.2
END DESCRIPTION:
XS GIS Cut Line= 3
      2367985.57      7040880.55      2368118.36      7040817.74
      2368393.04      7040814.15
#Sta/Elev= 30
  4744.6  682.16  4753.2  681.84  4761.3  681.78  4778.5  680.58    4784  681.08
  4792.6  679.87  4801.3  679.45  4806.8  679.95    4824  678.82  4829.6  678.98
  4846.8  678.35  4852.3  678.49  4875.1  677.59  4902.1  678.02  4922.1  677.74
  4952.1  676.09  4972.1  672.81  4982.1  669.77  5010.4  669.14  5013.9  669.14
  5014.1  669.64  5025.1  672.97  5032.2  675.32  5044.3  677.05  5052.2  677.49
  5062.2  677.47  5092.2  678.33  5132.2  680.98  5142.2  681.31  5166.2  681.35
#Mann= 5 ,-1 , 0
  4744.6     .05       0  4753.2    .075       0  4972.1     .04       0
  5025.1    .075       0  5044.3     .05       0
Bank Sta=4972.1,5025.1
XS Rating Curve= 0 ,0
Exp/Cntr=0.3,0.1

Type RM Length L Ch R = 1 ,13528   ,190,190,190
BEGIN DESCRIPTION:
Golf Course Creek Tr 1 37.0
END DESCRIPTION:
XS GIS Cut Line= 3
      2368051.92      7040941.61      2368166.83      7040878.77
       2368400.2       7040907.5
#Sta/Elev= 30
  4806.2  679.91  4826.5  679.33  4836.1  679.23  4857.9  678.36  4885.4  677.88
  4907.2  678.02  4916.8  678.24  4923.4  678.18  4929.1  677.78  4935.6   677.6
  4940.8   677.6  4949.4  676.87  4959.5  673.83  4969.6  670.55  4979.7  669.42
  4986.4  669.05  5028.3  668.32  5050.2  668.93  5060.3  671.25  5063.8  672.45
  5072.7  672.42  5080.4  674.22  5090.5  675.24  5100.6  677.05  5110.6  677.87
  5130.8  683.64  5140.9  684.76  5148.9  685.18  5153.9  685.05  5172.3  685.34
#Mann= 5 ,-1 , 0
  4806.2     .05       0  4826.5    .075       0  4986.4     .04       0
  5050.2    .075       0  5063.8     .05       0
Bank Sta=4986.4,5050.2
XS Rating Curve= 0 ,0
Exp/Cntr=0.3,0.1

Type RM Length L Ch R = 1 ,13338   ,219,219,219
BEGIN DESCRIPTION:
Golf Course Creek Tr 1 36.0
END DESCRIPTION:
XS GIS Cut Line= 3
      2368001.67      7041108.54        2368279.        7041060.
      2368480.93       7040982.9
#Sta/Elev= 30
  4723.2  682.38  4739.7   681.5  4744.8  681.75  4781.4  680.25  4799.2  679.21
  4804.3  679.24  4811.9  678.66  4832.2  677.84  4893.1  677.62  4923.5   676.6
  4928.6  676.01  4943.8  674.47    4954  672.91  4964.1  670.47  4972.5  669.76
  5067.2  669.14  5070.7  669.14    5071  669.64  5074.6  670.91  5079.9   671.7
  5099.3  676.58  5104.7  677.21  5111.8  679.33  5122.5  680.82  5129.4  681.38
  5154.1  682.12  5159.4   683.9    5176  684.22  5189.5  685.53  5220.9  685.65
#Mann= 4 ,-1 , 0
  4723.2     .05       0  4928.6    .075       0  4972.5    .033       0
    5071     .05       0
Bank Sta=4972.5,5071
XS Rating Curve= 0 ,0
Exp/Cntr=0.3,0.1

Type RM Length L Ch R = 1 ,13119   ,93,93,93
BEGIN DESCRIPTION:
Golf Course Creek Tr 1 35.4
END DESCRIPTION:
XS GIS Cut Line= 4
      2368008.85      7041280.86        2368323.      7041275.47
      2368495.32      7041176.75      2368544.34       7041085.7
#Sta/Elev= 30
  4596.3  683.14  4616.5  683.13  4636.5  682.52  4656.5   680.9  4666.5  680.48
  4696.5  678.33  4716.5  677.35  4726.5  676.64  4746.5  676.09  4756.5   676.1
  4786.5  675.25  4806.5  675.12  4818.8  674.59  4836.5  673.56  4846.5  671.99
  4856.5  669.94  4947.2  668.19  5072.7  669.35  5088.5  673.27  5101.8  675.06
  5116.8  676.29  5130.6  678.16  5146.8  679.81  5152.5  679.78  5162.2  680.15
  5168.7  680.77  5190.6  681.18  5196.3  680.82  5206.9  681.05  5212.5  680.77
#Mann= 4 ,-1 , 0
  4596.3     .05       0  4818.8    .075       0  4856.5    .033       0
  5072.7     .05       0
Bank Sta=4856.5,5072.7
XS Rating Curve= 0 ,0
Exp/Cntr=0.3,0.1

Type RM Length L Ch R = 1 ,13026   ,66,66,66
BEGIN DESCRIPTION:
Golf Course Creek Tr 1 35.2
END DESCRIPTION:
XS GIS Cut Line= 5
      2368010.68      7041311.38      2368265.56      7041350.86
      2368378.64      7041325.73      2368461.37      7041307.03
      2368744.56       7041169.5
#Sta/Elev= 30
  4574.1  683.14  4612.9  682.99    4623  680.74  4643.2  680.68  4665.8  679.71
  4683.7  677.31    4704   675.7  4764.7  674.38  4791.8  672.89  4796.9  673.69
  4952.3  673.92  4968.7  672.53    4979  670.18  4987.2  669.62  4987.5  669.12
    4991  669.12  4991.2  669.62  4995.5  670.96  5000.6  670.93  5009.7  672.64
    5020  673.09  5096.7  674.01  5104.2  673.53  5109.7  674.13    5217  674.25
  5245.1   677.2  5252.4  678.79  5267.6  679.66  5284.6  680.33  5347.5  680.88
#Mann= 3 ,-1 , 0
  4574.1     .05       0  4987.2    .033       0  4991.2     .05       0
Bank Sta=4987.2,4991.2
XS Rating Curve= 0 ,0
Exp/Cntr=0.3,0.1

Type RM Length L Ch R = 1 ,12960   ,157,157,157
BEGIN DESCRIPTION:
Golf Course Creek Tr 1 35.0
END DESCRIPTION:
XS GIS Cut Line= 4
      2368046.57      7041370.61       2368358.9      7041386.76
      2368457.62      7041377.79      2368719.73      7041318.55
#Sta/Elev= 30
  4616.4  680.54  4648.9  679.66  4668.9  677.85  4702.7  677.64    4719  675.75
    4739  674.91  4799.1  673.41  4829.1  673.69  4919.2  672.05  4931.7  671.31
  4946.5  669.01  4951.5  669.37  4959.4   667.1  4969.4  665.54  4977.5  665.07
  4977.7  664.57  4981.2  664.57  4981.5  665.07  5009.6  666.44  5019.6  665.67
  5026.5  669.15  5031.6  669.15    5043   672.4  5050.2  672.82  5172.6  674.75
    5245  674.42  5255.2  675.01  5269.2  676.84  5275.7  678.49    5297  681.49
#Mann= 3 ,-1 , 0
  4616.4     .05       0  4977.5    .033       0  4981.5     .05       0
Bank Sta=4977.5,4981.5
XS Rating Curve= 0 ,0
Exp/Cntr=0.3,0.1

Type RM Length L Ch R = 1 ,12803   ,151,151,151
BEGIN DESCRIPTION:
Golf Course Creek Tr 1 34.0
END DESCRIPTION:
XS GIS Cut Line= 3
      2368035.53      7041393.93      2368431.99      7041535.75
      2368721.06      7041635.32
#Sta/Elev= 30
  4678.7  678.79  4684.8  677.74  4771.8  676.02    4828   673.4  4852.3  673.31
  4858.8  672.33  4864.1  673.14  4889.6  671.09  4894.9  672.16  4915.1  670.59
  4920.4  672.14  4945.8  669.82  4951.1  672.06  4976.6  668.99  4981.9  669.71
  5010.7  663.55  5010.9  663.05  5014.7  663.55  5038.2     665  5043.5  666.59
  5063.6   667.9  5068.9  669.41  5094.4  667.89  5098.6  668.79  5125.6  668.18
  5297.6  674.56  5338.8  679.07    5361  680.12    5370  684.13  5405.5   683.9
#Mann= 3 ,-1 , 0
  4678.7     .05       0  5010.7    .033       0  5014.7     .05       0
Bank Sta=5010.7,5014.7
XS Rating Curve= 0 ,0
Exp/Cntr=0.3,0.1

Type RM Length L Ch R = 1 ,12652   ,229,229,229
BEGIN DESCRIPTION:
Golf Course Creek Tr 1 33.8
END DESCRIPTION:
XS GIS Cut Line= 3
      2367942.07       7041513.2      2368338.51      7041655.02
      2368628.64      7041754.95
#Sta/Elev= 30
  4589.1   677.9  4660.2  675.06  4710.6  674.54  4766.4   672.3  4777.5  671.23
  4819.5  669.29  4872.6  665.33    4926  663.18  4946.2  662.92  4966.2  661.03
  4966.4  660.53  4969.9  660.53  4970.2  661.03  4982.3  661.15  5031.8  663.51
    5053  663.69  5070.2  664.67  5075.5  664.26    5127  665.98  5132.6  666.74
  5163.8  667.52  5189.8  669.53    5195  669.03    5221   670.7  5226.3     670
  5252.2  672.35  5257.5  671.79  5283.4  673.66  5288.7  672.94    5317  675.24
#Mann= 3 ,-1 , 0
  4589.1     .05       0  4966.2    .033       0  4970.2     .05       0
Bank Sta=4966.2,4970.2
XS Rating Curve= 0 ,0
Exp/Cntr=0.3,0.1

Type RM Length L Ch R = 1 ,12423   ,182,182,182
BEGIN DESCRIPTION:
Golf Course Creek Tr 1 33.0
END DESCRIPTION:
XS GIS Cut Line= 3
      2367816.31      7041870.97      2368367.52      7041880.64
      2368670.55      7041745.25
#Sta/Elev= 30
  4487.6  675.19  4500.3  675.18  4540.3  673.59  4600.3  672.92  4820.3  665.59
  4900.4  662.18  4910.4  661.33  4940.4  660.36  4960.4  660.75  4978.4  660.13
  4978.6  659.63  4982.1  659.63  4982.4  660.13  5010.4  660.36  5030.4  661.26
  5049.4  661.02  5067.4  661.91    5078  661.95  5090.8  662.83  5101.3  663.86
  5139.1  665.95  5182.9  667.79  5199.6  669.32    5246  671.29  5251.5  671.05
  5314.3   673.9  5336.2  675.34  5349.8  676.75  5358.1  678.25  5370.8  679.14
#Mann= 5 ,-1 , 0
  4487.6     .05       0  4978.4    .033       0  4982.4     .05       0
  5067.4     .12       0  5090.8     .05       0
Bank Sta=4978.4,4982.4
XS Rating Curve= 0 ,0
Exp/Cntr=0.3,0.1

Type RM Length L Ch R = 1 ,12241   ,254,254,254
BEGIN DESCRIPTION:
Golf Course Creek Tr 1 32.0
END DESCRIPTION:
XS GIS Cut Line= 3
      2368129.02      7042309.98        2368429.        7042010.
      2368729.04      7041759.97
#Sta/Elev= 30
  4584.1  670.21  4626.5  668.66  4668.9  668.19  4711.4  666.98  4753.8  664.98
  4824.5   660.9  4838.6  660.68  4866.9  660.89  4881.1  660.29  4964.2  659.56
  5050.6  660.23  5058.5  661.75    5065  662.36  5072.8  663.79  5079.3  664.61
  5122.2  667.37  5128.7   667.2  5171.7  668.66  5220.8  671.74  5256.3  672.77
  5270.6  673.85  5278.4   674.8  5307.1  676.36  5313.6  676.26  5334.4  677.42
  5342.2   678.3  5348.7  678.12  5377.4  681.44  5395.6  684.36  5398.9  684.36
#Mann= 4 ,-1 , 0
  4584.1     .05       0  4881.1    .033       0  5050.6     .05       0
  5220.8     .05       0
Bank Sta=4881.1,5050.6
XS Rating Curve= 0 ,0
Exp/Cntr=0.3,0.1

Type RM Length L Ch R = 1 ,11987   ,234,234,234
BEGIN DESCRIPTION:
Golf Course Creek Tr 1 31.0
END DESCRIPTION:
XS GIS Cut Line= 3
        2368279.        7042460.        2368579.        7042210.
      2368828.99      7041910.02
#Sta/Elev= 30
  4609.7  670.09  4631.2  670.09  4659.8  669.26  4687.8  667.68  4709.3  667.17
  4744.4  664.85  4752.2  665.98  4773.1  666.16  4779.6  664.91  4793.9  663.33
    4816  662.12  4836.8  660.36  5104.5  659.43  5120.6   660.2  5142.7  662.17
  5156.4  662.73  5182.5  664.96  5192.3  665.63  5198.7  665.69  5206.5  666.91
  5220.8   668.2  5227.4  668.33  5241.7  669.72    5256  670.35  5284.6  673.22
  5305.5  674.53  5319.8  676.17  5340.6  677.47  5362.7  679.58  5390.7  681.13
#Mann= 5 ,-1 , 0
  4609.7     .05       0  4836.8    .033       0  5120.6     .05       0
  5182.5     .12       0  5192.3     .05       0
Bank Sta=4836.8,5120.6
XS Rating Curve= 0 ,0
Exp/Cntr=0.3,0.1

Type RM Length L Ch R = 1 ,11753   ,285,285,285
BEGIN DESCRIPTION:
Golf Course Creek Tr 1 30.0
END DESCRIPTION:
XS GIS Cut Line= 3
      2368228.99      7042910.01        2368779.        7042310.
      2368879.01      7042009.98
#Sta/Elev= 30
  4186.5   689.6  4189.9   689.6  4193.6  682.72  4200.4  684.14  4207.8   680.8
  4214.6  680.83  4236.2  679.19  4292.9  677.58  4313.8  677.52  4370.6  674.08
  4419.9  673.54  4455.7  672.13    4526  671.88  4590.1  670.13  4611.1  669.45
  4646.8  666.56    4661  666.78  4667.8  667.72    4682  668.36  4702.9  665.38
  4745.5  664.32    4788  660.47  5104.1  659.49  5126.9   660.1  5137.5  660.65
    5148  662.09  5169.1  662.91  5274.5  671.88  5295.6  673.07  5316.7  675.32
#Mann= 3 ,-1 , 0
  4186.5     .05       0    4788    .033       0  5126.9     .05       0
Bank Sta=4788,5126.9
XS Rating Curve= 0 ,0
Exp/Cntr=0.3,0.1

Type RM Length L Ch R = 1 ,11468   ,140,140,140
BEGIN DESCRIPTION:
Golf Course Creek Tr 1 29.0
END DESCRIPTION:
XS GIS Cut Line= 3
      2368429.01      7042959.99        2369029.        7042410.
      2369079.01      7042109.96
#Sta/Elev= 30
  4185.8  679.96  4242.2  677.49    4278  676.67  4327.3   674.3  4348.6  672.66
  4419.2  669.83  4426.6  668.78  4454.9  666.95  4483.3  667.21  4497.5  668.81
  4504.3  669.08  4511.4  668.79  4532.6  666.09  4553.6  665.04  4567.8  664.76
  4575.2  663.88    4582  663.98  4603.5  663.21  4624.5  663.27  4646.1  661.53
    4688  660.35  5038.5  659.62  5154.3  660.21  5182.2  662.01  5202.5  662.88
  5253.2  666.89  5270.9  668.85    5276  668.78  5283.6  669.58  5303.9  670.78
#Mann= 3 ,-1 , 0
  4185.8     .05       0    4688    .033       0  5154.3     .05       0
Bank Sta=4688,5154.3
XS Rating Curve= 0 ,0
Exp/Cntr=0.3,0.1

Type RM Length L Ch R = 1 ,11328   ,89,89,89
BEGIN DESCRIPTION:
Golf Course Creek Tr 1 28.4
END DESCRIPTION:
XS GIS Cut Line= 3
      2368718.83      7042979.81      2369099.21      7042573.65
       2369298.4      7042133.49
#Sta/Elev= 30
  4372.9  669.97    4401   668.6  4429.3  668.61  4443.5  668.22  4450.8  668.78
  4457.7  667.78  4500.1  664.93  4535.8  663.82  4599.3  660.43  4613.5  660.21
  4894.6   659.5  5164.3  660.08  5174.9  660.83  5196.8  660.69    5205  660.88
  5210.5   661.6  5228.1  662.69  5251.2  663.11  5273.6  664.21  5295.6  664.77
  5302.9  666.03  5308.4  666.01  5331.5  667.07  5349.1  667.03  5361.4  667.37
  5377.7  667.85  5383.4  668.34  5394.4  668.41  5400.8     669  5412.5  669.21
#Mann= 3 ,-1 , 0
  4372.9     .05       0  4613.5    .033       0  5164.3     .05       0
Bank Sta=4613.5,5164.3
XS Rating Curve= 0 ,0
Exp/Cntr=0.3,0.1

Type RM Length L Ch R = 1 ,11239   ,131,131,131
BEGIN DESCRIPTION:
Golf Course Creek Tr 1 28.2
END DESCRIPTION:
XS GIS Cut Line= 3
      2368812.33      7042976.57      2369192.68      7042570.43
      2369392.51      7042128.87
#Sta/Elev= 30
  4445.5   669.4  4468.8  666.48  4553.8  662.87  4561.1  664.25    4568  662.53
  4589.4  663.68  4596.3  662.38  4603.6  664.35  4610.5  662.17  4617.8   663.8
  4638.8  662.28  4646.1   664.1    4653  662.28  4667.1  664.97  4702.3  663.59
  4780.4   665.5    4844  663.81  4851.3  665.46  4872.3  663.85  4886.4  665.57
  5081.3  665.38    5189  663.85  5223.4  659.06  5223.7  658.56  5227.4  659.06
  5271.6  662.91  5323.3   663.2    5429  668.15  5465.2  669.18  5486.6  670.46
#Mann= 5 ,-1 , 0
  4445.5     .05       0  5223.4    .033       0  5227.4     .05       0
    5429     .12       0  5465.2     .05       0
Bank Sta=5223.4,5227.4
XS Rating Curve= 0 ,0
Exp/Cntr=0.3,0.1

Type RM Length L Ch R = 1 ,11108   ,201,201,201
BEGIN DESCRIPTION:
Golf Course Creek Tr 1 28.0
END DESCRIPTION:
XS GIS Cut Line= 3
      2368863.92      7043079.69      2369244.25      7042673.57
      2369443.35      7042233.63
#Sta/Elev= 30
  4465.6  669.74  4468.9  668.46    4483  666.75  4532.8  665.14  4561.1  663.11
  4638.9  659.74  4645.7  658.81  4752.2  654.87  4822.5  650.63  4941.2  647.27
  4941.4  646.77  4945.2  647.27  4957.3  648.23  4964.2   647.5  5006.7  647.59
  5124.7  654.56  5170.5  654.99  5188.1  655.84  5193.6  655.31  5211.2  656.01
  5239.8  655.51  5256.4  656.31  5268.4  655.68  5291.5  657.12  5322.3  656.93
  5360.8  659.75  5399.7  660.79  5435.6  661.64  5481.8  664.69  5504.9  665.11
#Mann= 4 ,-1 , 0
  4465.6     .05       0  4941.2    .033       0  4945.2     .05       0
  5399.7     .12       0
Bank Sta=4941.2,4945.2
XS Rating Curve= 0 ,0
Exp/Cntr=0.3,0.1

Type RM Length L Ch R = 1 ,10907   ,228,228,228
BEGIN DESCRIPTION:
Golf Course Creek Tr 1 27.0
END DESCRIPTION:
XS GIS Cut Line= 3
      2369078.98      7043110.02        2369379.        7042810.
      2369752.68      7042223.65
#Sta/Elev= 30
  4580.8  660.68    4694  655.21  4750.5  650.72  4835.4  647.16  5026.2  646.59
  5033.9   647.1  5049.1  648.08  5112.6  647.11  5121.9  648.24  5127.8  647.16
  5143.1  648.91    5149  648.38  5164.2  649.48  5206.7  649.91  5273.4  652.09
    5331  651.53  5367.3  652.11  5373.3  653.49  5382.6  653.26  5388.5  654.87
    5419  653.75  5446.1  654.34  5467.6  656.38  5485.6  656.61  5564.6  659.59
  5612.8   661.1  5621.7   662.1  5657.3  662.53  5692.9  664.94  5700.4  664.66
#Mann= 5 ,-1 , 0
  4580.8     .12       0  4835.4    .033       0  5033.9     .05       0
  5485.6     .12       0  5564.6     .05       0
Bank Sta=4835.4,5033.9
XS Rating Curve= 0 ,0
Exp/Cntr=0.3,0.1

Type RM Length L Ch R = 1 ,10679   ,343,343,343
BEGIN DESCRIPTION:
Golf Course Creek Tr 1 26.0
END DESCRIPTION:
XS GIS Cut Line= 3
      2369150.79      7043331.11        2369529.        7042960.
      2370039.26      7042413.71
#Sta/Elev= 30
  4465.1  664.94    4500  662.89  4535.3  661.57  4577.7  658.71  4655.6  655.52
  4733.3  650.72  4747.5  649.38  4789.9  647.58  5106.3  646.44  5122.2  647.11
  5136.4  649.09  5186.2  649.62  5214.1  650.99  5249.7  651.61  5368.1  656.74
  5391.4   657.9  5412.4  658.17  5500.4  657.05  5568.2  656.35  5610.7  655.04
  5652.8  655.06  5662.2  655.66  5674.3  656.67  5681.1  658.41  5688.4  658.78
  5695.3  660.91  5702.6  661.58  5730.9  665.67  5737.8  666.28  5742.5  665.27
#Mann= 6 ,-1 , 0
  4465.1     .12       0  4789.9    .033       0  5122.2     .05       0
  5368.1      .1       0  5500.4    .075       0  5662.2      .1       0
Bank Sta=4789.9,5122.2
XS Rating Curve= 0 ,0
Exp/Cntr=0.3,0.1

Type RM Length L Ch R = 1 ,10336   ,409,409,409
BEGIN DESCRIPTION:
Golf Course Creek Tr 1 25.0
END DESCRIPTION:
XS GIS Cut Line= 3
      2369429.01      7043509.99        2369729.        7043210.
      2370229.02      7042609.98
#Sta/Elev= 30
  4580.8  659.49  4609.1  657.74  4665.6  655.28  4736.4  650.86  4835.3  647.18
  4946.7  646.25  5225.7  647.76  5232.2  648.59  5267.3  650.73  5289.5  651.55
  5303.8  652.87  5338.9   654.5  5353.3  654.86  5388.4  654.23  5529.3  656.86
  5601.9  658.14  5643.5  658.21  5651.3  659.61  5657.9  659.82  5665.7  660.97
  5672.2  661.12    5680  662.23  5686.5   662.4  5694.3  663.85  5700.8  664.29
  5764.6  671.79  5772.4  673.12  5778.9  673.58  5782.8  674.54  5786.1  674.54
#Mann= 4 ,-1 , 0
  4580.8     .12       0  4835.3    .033       0  5225.7     .05       0
  5529.3      .1       0
Bank Sta=4835.3,5225.7
XS Rating Curve= 0 ,0
Exp/Cntr=0.3,0.1

Type RM Length L Ch R = 1 ,9927    ,105,105,105
BEGIN DESCRIPTION:
Golf Course Creek Tr 1 24.0
END DESCRIPTION:
XS GIS Cut Line= 4
      2369502.12      7043698.57      2369850.23      7043585.76
      2370001.72      7043521.29      2370220.93      7043140.91
#Sta/Elev= 30
  4556.3  662.17  4616.1  659.59  4647.6   657.1  4658.1   656.8  4728.3  652.73
  4733.5  651.96  4752.8  650.92  4760.3  650.35  4765.5  649.37  4792.2  647.54
  4795.5  646.99  4795.8  646.49  5194.8  647.39  5247.9  647.99  5253.7  649.57
  5269.5  650.99  5275.2  651.94  5328.4   653.2  5334.1  654.06  5349.9  654.21
  5355.7  654.81  5387.3  655.77    5393  656.72  5408.8  656.65  5414.6  657.55
  5430.4  657.73  5436.1  658.45  5451.9  658.66  5473.5  659.98  5525.9  661.14
#Mann= 3 ,-1 , 0
  4556.3     .05       0  4792.2    .033       0  5247.9     .05       0
Bank Sta=4792.2,5247.9
XS Rating Curve= 0 ,0
Exp/Cntr=0.3,0.1

Type RM Length L Ch R = 1 ,9822    ,121,121,121
BEGIN DESCRIPTION:
Golf Course Creek Tr 1 23.5
END DESCRIPTION:
XS GIS Cut Line= 4
      2369553.64      7043763.05      2369995.28      7043640.55
      2370159.66      7043434.26      2370314.21      7043167.02
#Sta/Elev= 30
  4610.8  661.14  4657.9  658.21  4715.3  656.11  4754.8  655.88  4789.1  654.94
    4866  654.51  4866.3  654.01  4869.8  654.01    4870  654.51  5031.5  655.75
  5135.7  655.85  5164.5  655.65  5178.9  654.96  5228.6  655.31  5271.8  654.87
  5364.1  655.74  5401.4  656.95  5407.2  657.97  5417.2  658.06  5422.9  658.95
  5460.3  660.34  5481.8   661.7  5497.6  661.46  5524.9  663.07  5540.6  662.66
  5546.4  663.18  5556.4  663.13  5562.2  663.89  5605.3  664.52  5641.6  665.69
#Mann= 3 ,-1 , 0
  4610.8     .05       0    4866    .033       0    4870     .05       0
Bank Sta=4866,4870
XS Rating Curve= 0 ,0
Exp/Cntr=0.3,0.1

Type RM Length L Ch R = 1 ,9701    ,203,203,203
BEGIN DESCRIPTION:
Golf Course Creek Tr 1 23.0
END DESCRIPTION:
XS GIS Cut Line= 3
      2369608.44       7043853.3      2370024.29      7043753.37
      2370335.44      7043512.79
#Sta/Elev= 30
  4621.6  662.74  4755.9  654.37  4781.7  652.04  4867.5  643.98  4879.3  641.51
  4899.9  639.69    4941  633.62  4990.4  633.14  4990.7  632.64  4994.4  633.14
  4998.5  634.31  5003.7  633.34  5028.6  635.38  5040.5   637.3  5045.6  636.35
  5049.1  637.73  5062.3  638.79  5097.6  639.75  5180.6  644.63  5211.8  646.79
  5226.2  647.39  5232.5   649.7  5240.7  650.15  5255.2  647.26  5269.7  646.56
  5296.8  653.36  5339.5  655.48  5375.6  659.11  5410.9  660.49  5442.6  662.89
#Mann= 8 ,-1 , 0
  4621.6     .12       0  4781.7     .05       0  4990.4    .033       0
  4994.4     .05       0  5028.6     .12       0  5180.6     .05       0
  5211.8     .12       0  5339.5     .05       0
Bank Sta=4990.4,4994.4
XS Rating Curve= 0 ,0
Exp/Cntr=0.3,0.1

Type RM Length L Ch R = 1 ,9498    ,182,182,182
BEGIN DESCRIPTION:
Golf Course Creek Tr 1 22.7
END DESCRIPTION:
XS GIS Cut Line= 3
      2369627.83      7044017.68      2369972.71      7043972.55
      2370739.83      7043650.23
#Sta/Elev= 30
  4599.8  667.63  4691.7   662.5    4771  655.89  4812.8  654.03  4854.9  650.62
  4968.9  639.44  4976.1  637.92  4992.7  631.94  5006.7  631.82  5006.9  631.32
  5010.7  631.82  5016.4   634.1  5030.4  636.17  5062.9  635.21  5069.4  631.94
  5106.3  637.04  5193.1   639.8  5244.9     644    5269  644.48  5275.7  645.66
  5353.5  650.32  5511.1  652.99  5594.4  653.36  5605.3  653.27  5611.6  651.81
    5617  652.59  5626.9   650.6  5670.3  649.83  5717.5  656.53  5779.7  661.75
#Mann= 5 ,-1 , 0
  4599.8     .12       0  5006.7     .07       0  5010.7     .12       0
  5244.9     .05       0  5353.5      .1       0
Bank Sta=5006.7,5010.7
XS Rating Curve= 0 ,0
Exp/Cntr=0.3,0.1

Type RM Length L Ch R = 1 ,9316    ,172,172,172
BEGIN DESCRIPTION:
Golf Course Creek Tr 1 22.4
END DESCRIPTION:
XS GIS Cut Line= 3
      2369705.18      7044172.39      2370050.07      7044127.27
      2370815.52      7043805.65
#Sta/Elev= 30
  4578.9   663.2  4663.4  657.34  4764.3  648.61  4784.5  647.87  4863.6  640.59
    4961  636.11  5001.5  632.86  5008.5  630.92  5030.2  630.57  5030.5  630.07
  5034.2  630.57  5055.7  631.75  5061.4  633.51  5066.8  632.78  5084.8  637.49
  5243.6  644.41  5323.2  647.93  5391.9  651.83  5479.4  652.34  5556.1  651.01
  5574.5  654.99  5579.9  653.74  5587.2  656.86  5603.6  657.83  5609.1  655.47
  5632.8  655.29  5695.7  657.79  5712.8  662.68  5724.5  663.29    5757  663.99
#Mann= 8 ,-1 , 0
  4578.9     .05       0  5030.2    .033       0  5034.2     .05       0
  5084.8     .12       0  5243.6     .05       0  5323.2      .1       0
  5712.8     .05       0  5724.5      .1       0
Bank Sta=5030.2,5034.2
XS Rating Curve= 0 ,0
Exp/Cntr=0.3,0.1

Type RM Length L Ch R = 1 ,9144    ,315,315,315
BEGIN DESCRIPTION:
Golf Course Creek Tr 1 22.0
END DESCRIPTION:
XS GIS Cut Line= 3
      2369772.82      7044330.34      2370108.09       7044256.2
      2370478.96      7044210.01
#Sta/Elev= 30
  4585.1  661.88  4608.3  657.94  4613.4  658.02  4657.1  654.09  4673.4  651.82
  4744.4  648.99  4765.5  647.21  4793.1  643.86  4841.9  641.62  4885.5  636.88
  4890.6  637.12  4926.4  634.36  4936.3  634.12  4941.3  634.96  4969.7  633.28
  4979.8  630.84  4997.9  629.44  4998.2  628.94  5001.7  628.94  5001.9  629.44
    5010  629.57  5022.1  631.21  5030.2  633.33  5090.6  639.31  5110.8  642.32
  5183.6  647.25  5211.5   650.1  5264.4  657.28  5282.1  658.91  5302.2  659.59
#Mann= 3 ,-1 , 0
  4585.1     .05       0  4997.9     .05       0  5001.9     .05       0
Bank Sta=4997.9,5001.9
XS Rating Curve= 0 ,0
Exp/Cntr=0.3,0.1

Type RM Length L Ch R = 1 ,8829    ,327,327,327
BEGIN DESCRIPTION:
Golf Course Creek Tr 1 21.0
END DESCRIPTION:
XS GIS Cut Line= 3
      2369950.14      7044626.88      2370375.62      7044481.83
      2370654.98      7044391.92
#Sta/Elev= 30
  4652.6  656.09  4688.9  653.87  4694.2  652.92  4704.2  652.81  4751.6   649.6
    4809  646.91  4852.1  642.09  4894.4  638.41  4934.4  632.52  4947.2  628.44
  4955.8  628.16    4956  627.66  4959.5  627.66  4959.8  628.16  4989.5  628.81
    4997  628.41  5010.6  630.33  5021.2  630.68  5028.4  631.91  5084.6  633.91
  5096.4   635.6  5101.3     637  5116.2  638.06  5122.9  639.89  5147.7   642.5
  5219.2  648.69  5242.2  650.03  5315.4   658.2  5352.7   661.5  5395.6  663.18
#Mann= 3 ,-1 , 0
  4652.6     .05       0  4955.8    .033       0  4959.8     .05       0
Bank Sta=4955.8,4959.8
XS Rating Curve= 0 ,0
Exp/Cntr=0.3,0.1

Type RM Length L Ch R = 1 ,8502    ,381,381,381
BEGIN DESCRIPTION:
Golf Course Creek Tr 1 20.0
END DESCRIPTION:
XS GIS Cut Line= 3
      2370033.97      7044868.62        2370379.        7044810.
      2370777.06      7044624.34
#Sta/Elev= 30
    4654  656.07  4659.1  655.19    4680  654.12  4735.2  649.11  4740.3  649.21
  4780.8  645.91  4821.4  643.38  4841.7  640.55  4892.4  635.53    4911  632.99
  4916.1  633.24  4922.8  632.66    4933  630.12  4951.3  628.19  4951.5  627.69
    4955  627.69  4955.3  628.19  4976.4  629.07  4993.8  628.23  5012.6  628.47
  5018.2  629.25    5026  631.33  5115.1  634.76  5235.7   642.1  5275.2   643.9
  5280.7  644.69  5320.9  646.08  5349.3  648.06  5389.5  649.23  5443.2  651.84
#Mann= 3 ,-1 , 0
    4654     .05       0  4951.3    .033       0  4955.3     .05       0
Bank Sta=4951.3,4955.3
XS Rating Curve= 0 ,0
Exp/Cntr=0.3,0.1

Type RM Length L Ch R = 1 ,8121    ,350,350,350
BEGIN DESCRIPTION:
Golf Course Creek Tr 1 19.0
END DESCRIPTION:
XS GIS Cut Line= 3
      2370043.64      7045232.85        2370379.        7045160.
        2370679.        7045010.
#Sta/Elev= 30
  4652.5  646.91  4735.7  641.69  4740.8  641.96  4779.7  639.48  4784.8  639.84
  4903.6  633.04  4913.8  631.44    4922  625.31  4927.1  627.46  4934.3  624.96
  4954.8  621.95    4965  623.39  4971.1  626.41  4985.5  625.44  4993.1  622.66
  4998.5  622.66  5009.7  620.34  5024.4  618.88  5024.7  618.38  5028.4  618.88
  5048.8  620.19  5093.5  627.06  5129.8  628.88  5138.2  629.99  5152.2  629.89
  5174.6   631.5  5196.9  635.22  5219.3  633.46    5250  637.55  5331.1  643.86
#Mann= 3 ,-1 , 0
  4652.5     .05       0  5024.4    .033       0  5028.4     .05       0
Bank Sta=5024.4,5028.4
XS Rating Curve= 0 ,0
Exp/Cntr=0.3,0.1

Type RM Length L Ch R = 1 ,7771    ,439,439,439
BEGIN DESCRIPTION:
Golf Course Creek Tr 1 18.0
END DESCRIPTION:
XS GIS Cut Line= 3
      2370043.58      7045535.85      2370614.15      7045442.36
      2370828.97      7045310.02
#Sta/Elev= 30
    4508  652.52  4543.9  649.64  4577.2  648.22  4633.5  643.81  4736.4  637.78
  4761.2  635.96  4817.5  630.22  4827.6  629.75  4837.8  630.43  4871.8   626.8
  4939.1  624.04  4969.5  623.68  4979.6  621.78  4989.8  618.14  5009.6  617.68
  5009.8  617.18  5013.6  617.68  5030.3  618.62  5040.4  621.06  5060.7  623.13
    5081  626.69  5104.9  627.94  5149.6  631.75  5193.6  635.81  5221.1  636.71
  5236.2  636.07  5244.6  637.47  5257.5  641.28  5288.3  646.65  5338.5  652.69
#Mann= 5 ,-1 , 0
    4508     .05       0  4871.8     .12       0  5009.6     .07       0
  5013.6     .12       0  5149.6     .05       0
Bank Sta=5009.6,5013.6
XS Rating Curve= 0 ,0
Exp/Cntr=0.3,0.1

Type RM Length L Ch R = 1 ,7332    ,542,542,542
BEGIN DESCRIPTION:
Golf Course Creek Tr 1 17.0
END DESCRIPTION:
XS GIS Cut Line= 3
      2370162.85      7045961.32      2370736.63      7045825.93
      2370985.31      7045626.99
#Sta/Elev= 30
  4572.8  654.98  4597.4  650.18  4630.5  646.59  4671.6  643.91  4687.2  641.13
    4777  634.86  4814.2  629.68  4819.3  630.24  4846.3  626.61  4861.6  626.79
  4897.6  622.76  4918.2  617.63  4938.7  615.06  4986.6  613.88  4986.8  613.38
  4990.6  613.88  4993.7  614.99  5036.1  616.36  5078.4  619.95  5083.5   619.1
  5113.4  621.05    5134  623.61  5190.2  625.47  5267.8  631.98  5353.5  636.66
  5382.3  639.82  5388.7  637.94  5403.1  638.21  5423.9  640.57  5480.8  641.34
#Mann= 3 ,-1 , 0
  4572.8     .05       0  4986.6     .05       0  4990.6     .05       0
Bank Sta=4986.6,4990.6
XS Rating Curve= 0 ,0
Exp/Cntr=0.3,0.1

Type RM Length L Ch R = 1 ,6790    ,203,203,203
BEGIN DESCRIPTION:
Golf Course Creek Tr 1 16.0
END DESCRIPTION:
XS GIS Cut Line= 3
      2370259.55      7046499.61      2370959.04      7046273.97
      2371335.09      7046161.47
#Sta/Elev= 30
  4401.8  631.31    4481  628.92  4537.8  628.64  4656.1   624.2  4737.7  622.05
    4844  620.48  4902.9  617.23  4926.6  612.02    4967  606.64  4989.6  605.51
    4997   603.7  4997.3   603.2    5001   603.7  5004.3  605.24  5010.6  604.79
  5026.6  606.59  5036.3  607.35  5042.2   609.4  5068.4  613.51  5094.7  612.07
  5100.4  612.84  5105.7  612.33  5126.2  615.37  5147.2  617.19  5198.6  618.56
  5236.9  621.25  5260.7  621.08  5303.1  624.33  5355.9  626.62  5529.3  637.22
#Mann= 7 ,-1 , 0
  4401.8     .05       0  4656.1      .1       0  4737.7     .05       0
    4997    .033       0    5001     .05       0  5026.6    .075       0
  5260.7     .05       0
Bank Sta=4997,5001
XS Rating Curve= 0 ,0
Exp/Cntr=0.3,0.1

Type RM Length L Ch R = 1 ,6587    ,263,263,263
BEGIN DESCRIPTION:
Golf Course Creek Tr 1 15.0
END DESCRIPTION:
XS GIS Cut Line= 3
      2370572.24      7046657.54      2370975.15      7046438.36
      2371264.58      7046309.72
#Sta/Elev= 30
  4587.5  619.54  4700.4  619.21  4891.3   616.9  4907.5  616.32  4923.6  612.41
  4929.3  612.68  4959.5  610.51  4967.3  607.49  4982.3  603.21  4987.2  602.59
  4987.4  602.09  4990.9  602.09  4991.2  602.59    5011  607.19  5039.2  610.27
  5045.5  611.54  5050.3  611.54  5055.1  612.19  5072.3  615.34  5078.4   617.1
  5083.9  615.87  5101.7  617.85  5107.1  616.89  5176.9  619.93  5236.4   621.9
  5291.1  622.19  5298.6  625.39  5304.1  625.38  5321.9  628.93  5362.9  630.58
#Mann= 3 ,-1 , 0
  4587.5     .05       0  4987.2    .033       0  4991.2     .05       0
Bank Sta=4987.2,4991.2
XS Rating Curve= 0 ,0
Exp/Cntr=0.3,0.1

Type RM Length L Ch R = 1 ,6324    ,352,352,352
BEGIN DESCRIPTION:
Golf Course Creek Tr 1 14.0
END DESCRIPTION:
XS GIS Cut Line= 3
      2370672.16      7046886.39        2370979.        7046710.
      2371210.48      7046570.49
#Sta/Elev= 30
  4641.9  618.21  4783.8  616.46  4870.1  616.29    4892   615.5  4923.2   609.7
    4929   607.4  4938.2  605.15  4944.8  605.01  4960.6   601.3  4966.4  601.74
  4970.8  596.17    4971  595.67  4974.5  595.67  4974.8  596.17  4982.2  602.79
  5009.4  603.12  5046.3  605.51  5054.2  608.44  5067.7   611.6  5077.4  612.82
  5098.7  613.55  5104.6  614.47  5112.6  614.05    5157  614.84  5184.2  616.77
  5221.1  616.85  5236.6  619.91  5257.9  622.49  5262.3  624.24  5266.1  624.24
#Mann= 3 ,-1 , 0
  4641.9     .05       0  4970.8    .033       0  4974.8     .05       0
Bank Sta=4970.8,4974.8
XS Rating Curve= 0 ,0
Exp/Cntr=0.3,0.1

Type RM Length L Ch R = 1 ,5972    ,142,142,142
BEGIN DESCRIPTION:
Golf Course Creek Tr 1 13.0
END DESCRIPTION:
XS GIS Cut Line= 3
      2370992.21      7047144.48        2371179.        7046960.
      2371284.98      7046800.18
#Sta/Elev= 30
    4737  613.27  4808.6  613.69  4865.2  612.27  4886.4  608.63  4914.7  605.24
  4928.9  605.11  4935.9  606.53    4943  605.77    4950  606.31  4957.2  604.92
  4978.3  596.88    4994  595.24  4994.3  594.74    4998  595.24  5007.1  596.18
  5013.1  599.39  5022.1  602.47  5028.1  606.98  5043.2  607.22  5049.2  608.99
  5058.2  609.39  5064.2  610.75  5079.2  611.04  5115.3  616.45  5121.3  616.34
  5130.4  618.73  5136.4  617.73  5148.9  619.29  5155.1   618.9  5191.3  620.24
#Mann= 5 ,-1 , 0
    4737     .05       0    4994    .033       0    4998     .05       0
  5148.9    .075       0  5155.1     .05       0
Bank Sta=4994,4998
XS Rating Curve= 0 ,0
Exp/Cntr=0.3,0.1

Type RM Length L Ch R = 1 ,5830    ,87,87,87
BEGIN DESCRIPTION:
Golf Course Creek Tr 1 12.8
END DESCRIPTION:
XS GIS Cut Line= 3
      2371067.76      7047355.99      2371186.96      7047134.38
      2371380.03      7046899.34
#Sta/Elev= 30
  4682.3  608.59  4738.9  608.67  4842.8  605.15    4859  605.57  4870.8  606.61
  4902.9  605.75  4908.5   606.3  4916.2  605.69  4959.9  605.93  4966.4  604.31
  4974.2  604.37  4980.7  598.22  4990.1  594.09  5015.5  593.47  5030.2  594.97
  5038.1  601.09  5044.6  600.63  5052.5  605.03  5073.3  609.35  5108.4  612.36
  5130.7  613.43  5151.5  616.08  5180.2   618.2  5186.6  617.81    5196  618.25
    5201  618.03  5208.9  618.84  5215.3  620.17  5229.7  621.94  5238.1  621.64
#Mann= 4 ,-1 , 0
  4682.3     .05       0  4990.1     .04       0  5030.2     .05       0
    5196    .075       0
Bank Sta=4990.1,5030.2
XS Rating Curve= 0 ,0
Exp/Cntr=0.3,0.1

Type RM Length L Ch R = 1 ,5743    ,90,90,90
BEGIN DESCRIPTION:
Golf Course Creek Tr 1 12.6
END DESCRIPTION:
XS GIS Cut Line= 3
      2371114.78      7047371.07      2371307.82      7047107.52
      2371426.87       7046914.7
#Sta/Elev= 30
  4731.8  609.52  4749.6  608.98  4764.2  609.48  4785.1  608.06  4807.5  607.64
  4820.6  606.51  4900.1  604.83  4914.7  603.19  4920.9  601.06  4929.4  599.66
  4935.6  597.49  4956.5  594.87  4969.4  593.86  5029.8  594.72    5043  603.86
  5050.6  604.99  5058.5  605.19  5071.7  607.33  5079.1   610.3    5093  613.21
  5173.1  613.19  5181.7  613.71  5187.6  615.88  5196.6  616.99  5218.4  616.25
  5224.3  616.83  5231.9  619.45  5239.6  620.75  5263.1  623.03  5285.1  623.17
#Mann= 4 ,-1 , 0
  4731.8     .05       0  4956.5    .033       0  5029.8     .05       0
  5263.1    .075       0
Bank Sta=4956.5,5029.8
XS Rating Curve= 0 ,0
Exp/Cntr=0.3,0.1

Type RM Length L Ch R = 1 ,5653    ,114,114,114
BEGIN DESCRIPTION:
Golf Course Creek Tr 1 12.2
END DESCRIPTION:
XS GIS Cut Line= 3
      2371189.67      7047417.99      2371353.15      7047194.81
      2371497.59      7046960.85
#Sta/Elev= 30
  4701.3  609.37  4777.7  605.98  4821.6   605.5  4827.8  604.37  4885.7  604.12
  4898.9  603.66  4913.5  601.57  4928.2  598.77  4934.7  595.82  4947.3  593.71
  4978.4  594.78  4984.6  598.94    4993  600.17  4999.2   602.6  5013.9     604
  5027.8  603.26  5034.5  605.67  5057.1  606.46  5071.2  608.41  5083.3  611.34
  5092.5  613.43  5123.2  613.76  5144.5  612.89  5174.6  613.66  5183.9  614.72
  5187.1   615.4  5217.8  614.78  5223.7  618.27  5233.2  620.06  5252.9  620.87
#Mann= 6 ,-1 , 0
  4701.3     .05       0  4885.7    .075       0  4934.7    .033       0
  4978.4    .075       0  5083.3     .05       0  5183.9    .075       0
Bank Sta=4934.7,4978.4
XS Rating Curve= 0 ,0
Exp/Cntr=0.3,0.1

Type RM Length L Ch R = 1 ,5539    ,389,389,389
BEGIN DESCRIPTION:
Golf Course Creek Tr 1 12.0
END DESCRIPTION:
XS GIS Cut Line= 3
      2371237.34      7047523.79      2371430.36      7047260.28
      2371549.54      7047067.25
#Sta/Elev= 30
  4733.5  609.58  4742.4  609.13    4746  608.93  4824.1  609.19  4844.9  606.53
  4859.6  603.67  4886.9  604.24  4895.1   603.7  4901.3  602.89  4909.8   600.3
    4916  600.71  4930.6   596.7  4951.5  595.55  4973.7  596.82  4980.8  595.93
    4987  594.22  5008.4  593.15  5037.2  594.58  5045.6  598.66  5051.8  599.89
  5057.2  602.52    5088  604.79  5124.6   609.9  5203.8  609.68  5213.3  611.09
  5219.2   613.3  5248.5  612.28  5255.9  614.36  5261.8  617.02    5287  616.88
#Mann= 5 ,-1 , 0
  4733.5    .075       0  4742.4     .05       0    4746    .075       0
    4987    .033       0  5037.2    .075       0
Bank Sta=4987,5037.2
XS Rating Curve= 0 ,0
Exp/Cntr=0.3,0.1

Type RM Length L Ch R = 1 ,5150    ,350,350,350
BEGIN DESCRIPTION:
Golf Course Creek Tr 1 11.0
END DESCRIPTION:
XS GIS Cut Line= 3
      2371545.67      7047663.21        2371729.        7047460.
      2371938.89      7047141.06
#Sta/Elev= 30
  4721.6  613.21  4740.1  612.99  4747.5  613.43  4775.9  612.44  4782.7  610.98
  4790.1  610.13  4796.9  607.97  4818.5  605.03  4853.7  604.99  4874.6  603.54
  4882.1  602.28  4910.5  599.84  4924.7   596.4  4931.4  596.03  4953.1  593.45
  4965.5  592.91    5060  593.52  5067.1  596.09  5075.1  600.96  5090.2  601.82
  5096.2  601.49  5111.3  601.89  5118.1  602.64  5126.4     603  5132.3  603.91
  5210.8  604.75  5225.7  606.41  5255.9  606.66  5306.5  608.33  5377.1  611.77
#Mann= 4 ,-1 , 0
  4721.6     .05       0  4953.1    .033       0    5060     .05       0
  5118.1     .05       0
Bank Sta=4953.1,5060
XS Rating Curve= 0 ,0
Exp/Cntr=0.3,0.1

Type RM Length L Ch R = 1 ,4800    ,259,259,259
BEGIN DESCRIPTION:
Golf Course Creek Tr 1 10.0
END DESCRIPTION:
XS GIS Cut Line= 3
      2371648.16      7047944.01      2371996.93      7047666.42
      2372126.53       7047454.1
#Sta/Elev= 30
  4640.3  617.68  4644.5  616.18  4665.3  614.91  4673.3  613.06  4679.7  613.46
    4715  610.13    4723   608.8  4737.4  603.92  4765.5  604.32    4779  605.65
  4865.5  600.17  4886.3  602.52  4900.8  600.69    4936  600.44    4944  597.15
  4950.4  597.59  4964.8   595.8  5035.3  593.73  5040.4   593.2  5145.3   594.4
  5167.8  599.29  5268.5  603.21  5274.4  604.85    5284  604.89  5289.8  607.34
  5305.3  607.32  5311.2   610.5  5320.8  610.47  5326.6  612.53  5334.8  612.19
#Mann= 3 ,-1 , 0
  4640.3     .05       0  5035.3    .033       0  5145.3     .05       0
Bank Sta=5035.3,5145.3
XS Rating Curve= 0 ,0
Exp/Cntr=0.3,0.1

Type RM Length L Ch R = 1 ,4541    ,139,139,139
BEGIN DESCRIPTION:
Golf Course Creek Tr 1 9.6
END DESCRIPTION:
XS GIS Cut Line= 3
      2371774.56      7048043.53      2372058.17      7047930.73
      2372398.49      7047681.23
#Sta/Elev= 30
  4655.4  612.45  4660.5  612.45  4670.9  609.19  4692.5   609.7  4746.3  608.98
    4761  607.24  4778.6  604.08  4785.3  602.18  4790.7  602.32  4800.1  600.97
  4875.4  598.49  4907.7  598.65  4964.2   597.6  4983.7  593.35  4987.7  589.62
  4988.1  589.12  5104.9  589.93  5125.8  595.19  5134.2  596.59  5140.4  595.74
  5161.3  595.77  5190.6  597.05  5197.2  598.08  5205.3   601.5  5211.5  599.66
  5219.9   601.7  5226.1  601.14  5240.8  602.91  5305.6  604.69  5382.6  607.72
#Mann= 3 ,-1 , 0
  4655.4     .05       0  4987.7    .033       0  5104.9     .05       0
Bank Sta=4987.7,5104.9
XS Rating Curve= 0 ,0
Exp/Cntr=0.3,0.1

Type RM Length L Ch R = 1 ,4402    ,257,257,257
BEGIN DESCRIPTION:
Golf Course Creek Tr 1 9.4
END DESCRIPTION:
XS GIS Cut Line= 3
      2371900.22      7048108.02      2372183.88       7047995.2
      2372524.07      7047745.79
#Sta/Elev= 30
  4672.6  605.51  4729.2   604.2    4757  604.91  4787.6   602.4  4816.3  601.99
    4822  601.04  4832.7  597.33  4870.3  597.94  4940.3  597.03  4948.5  594.88
  4953.9  594.95  4961.9   589.2  4972.6  587.71  5007.4  587.03  5019.2  585.62
  5019.6  585.12  5023.6  585.62  5028.3  588.58  5049.1  590.79    5071  591.14
  5107.8  593.65  5164.1  595.75  5220.5  599.55    5257  604.35  5285.3  606.78
  5335.5   607.9    5371  606.83  5379.5     607  5385.7  608.72  5399.7  608.29
#Mann= 5 ,-1 , 0
  4672.6     .05       0  4729.2    .075       0  4787.6     .05       0
  5019.2     .05       0  5023.6     .05       0
Bank Sta=5019.2,5023.6
XS Rating Curve= 0 ,0
Exp/Cntr=0.3,0.1

Type RM Length L Ch R = 1 ,4145    ,297,297,297
BEGIN DESCRIPTION:
Golf Course Creek Tr 1 9.0
END DESCRIPTION:
XS GIS Cut Line= 3
      2371955.07       7048372.3      2372238.68      7048259.51
        2372579.        7048010.
#Sta/Elev= 30
  4595.7  609.21  4615.8  608.71  4640.1  606.95  4645.4  607.46  4675.3  604.14
  4738.1  600.02    4769   598.1  4879.7   591.3  4885.6  590.37  4904.2  589.47
    4908   588.6  4922.7  587.07  4958.2  585.68  5020.8  585.05  5021.2  584.55
  5024.8  584.55  5025.3  585.05  5037.7  585.19  5073.2  587.13    5094  589.08
  5108.7  591.36  5129.6  593.71  5150.4  595.56  5250.7  602.04  5259.2  603.77
  5265.4  603.95  5273.3  605.33  5286.3  606.34  5309.4  609.16  5322.9  610.04
#Mann= 5 ,-1 , 0
  4595.7     .05       0  4738.1    .075       0    4769     .05       0
  5020.8    .033       0  5025.3     .05       0
Bank Sta=5020.8,5025.3
XS Rating Curve= 0 ,0
Exp/Cntr=0.3,0.1

Type RM Length L Ch R = 1 ,3848    ,193,193,193
BEGIN DESCRIPTION:
Golf Course Creek Tr 1 8.3
END DESCRIPTION:
XS GIS Cut Line= 3
      2372158.05      7048604.41      2372351.49      7048559.27
      2372583.24      7048314.65
#Sta/Elev= 30
  4640.6  605.33  4672.4  601.08  4679.8  599.18  4684.9  599.63  4692.9  598.18
  4703.2  597.28  4727.4  597.18    4770  595.22  4785.3   595.4  4839.2  590.35
  4872.3  585.46  4907.5  584.85  4914.8  585.57  4921.7   584.8  4935.8  584.67
  4976.1  581.48  4976.5  580.98  4980.1  580.98  4980.6  581.48  4999.7  581.61
  5020.8  584.79  5028.1  586.48  5042.2  588.13  5049.1  588.56  5056.4  588.03
  5070.5  588.88  5077.4  591.14  5091.6  593.18  5127.2  594.23  5176.2  596.91
#Mann= 3 ,-1 , 0
  4640.6     .05       0  4976.1    .033       0  4980.6     .05       0
Bank Sta=4976.1,4980.6
XS Rating Curve= 0 ,0
Exp/Cntr=0.3,0.1

Type RM Length L Ch R = 1 ,3655    ,262,262,262
BEGIN DESCRIPTION:
Golf Course Creek Tr 1 8.0
END DESCRIPTION:
XS GIS Cut Line= 3
      2372229.05      7048649.52      2372483.65       7048604.4
      2372657.67      7048411.04
#Sta/Elev= 30
  4797.3  596.44  4817.6  594.76  4868.3  593.35  4876.9   591.9    4882  592.05
  4936.1  586.74  4941.1  586.88  4949.6  585.73  4959.7  585.38  4980.1  582.95
  4995.2  582.98  5000.4     582  5010.5   581.7    5047  581.39  5047.4  580.89
    5051  580.89  5051.5  581.39  5084.1  582.15  5090.8  583.39  5098.3  582.91
    5105  584.14  5112.5  583.47  5119.3  586.11  5126.7  585.59  5140.9  588.52
  5232.9  593.13  5239.6   593.8  5247.1  597.02  5253.8  598.84    5316  599.23
#Mann= 3 ,-1 , 0
  4797.3     .05       0    5047     .05       0  5051.5     .05       0
Bank Sta=5047,5051.5
XS Rating Curve= 0 ,0
Exp/Cntr=0.3,0.1
