--- Whites Branch.prj (project) ---

Proj Title=Whites Branch Base Level Engineering
Current Plan=p01
Default Exp/Contr=0.3,0.1
English Units
Geom File=g01
Flow File=f01
Plan File=p01
Y Axis Title=Elevation
X Axis Title(PF)=Main Channel Distance
X Axis Title(XS)=Station
BEGIN DESCRIPTION:
Whites Branch
END DESCRIPTION:
DSS Export Rating Curves= 0
DSS Export Rating Curve Sorted= 0
DSS Export Volume Flow Curves= 0
DXF OffsetX= 0
DXF OffsetY= 0
DXF ScaleX= 1
DXF ScaleY= 10

--- Whites Branch.p01 (plan) ---

Plan Title=Multiple Run
Short Identifier=Multiple
Geom File=g01
Flow File=f01
Subcritical Flow
K Sum by GR= 0
Std Step Tol= 0.01
Critical Tol= 0.01
Num of Std Step Trials= 20
Max Error Tol= 0.3
Flow Tol Ratio= 0.001
Split Flow NTrial= 30
Split Flow Tol= 0.02
Split Flow Ratio= 0.02
Log Output Level= 0
Friction Slope Method= 1
Unsteady Friction Slope Method= 2
Unsteady Bridges Friction Slope Method= 1
Parabolic Critical Depth
Global Vel Dist=  1 , 1 , 1
Global Log Level= 0
CheckData=True
Encroach Param= -1, 0, 0, 0
BEGIN DESCRIPTION:
Multiple Run
END DESCRIPTION:

--- Whites Branch.f01 (steady flow) ---

Flow Title=Multiple
Program Version=4.10
Number of Profiles= 7
Profile Names=10-year,25-year,50-year,1pct_min,100-year,1pct_plu,500-year
River Rch & RM=Whites Branch,Reach-1         ,35755
     236     304     357     209     417     832     569
River Rch & RM=Whites Branch,Reach-1         ,32515
     412     551     664     398     794    1584    1136
River Rch & RM=Whites Branch,Reach-1         ,31278
     610     835    1020     620    1236    2466    1817
River Rch & RM=Whites Branch,Reach-1         ,28459
     774    1071    1319     806    1607    3207    2394
River Rch & RM=Whites Branch,Reach-1         ,25664
     956    1339    1662    1022    2040    4070    3081
River Rch & RM=Whites Branch,Reach-1         ,23547
    1117    1576    1966    1215    2424    4836    3695
River Rch & RM=Whites Branch,Reach-1         ,20783
    1196    1690    2110    1304    2602    5193    3971
River Rch & RM=Whites Branch,Reach-1         ,14315
    2203    3204    4078    2566    5119   10214    8094
River Rch & RM=Whites Branch,Reach-1         ,9651
    2871    4210    5388    3406    6796   13560   10847
River Rch & RM=Whites Branch,Reach-1         ,5516
    3033    4452    5700    3604    7191   14348   11482
River Rch & RM=Whites Branch,Reach-1         ,254
    3184    4677    5993    3791    7564   15092   12090
Boundary for River Rch & Prof#=Whites Branch,Reach-1         , 1
Up Type= 0
Dn Type= 3
Dn Slope=0.0005
Boundary for River Rch & Prof#=Whites Branch,Reach-1         , 2
Up Type= 0
Dn Type= 3
Dn Slope=0.0005
Boundary for River Rch & Prof#=Whites Branch,Reach-1         , 3
Up Type= 0
Dn Type= 3
Dn Slope=0.0005
Boundary for River Rch & Prof#=Whites Branch,Reach-1         , 4
Up Type= 0
Dn Type= 3
Dn Slope=0.0005
Boundary for River Rch & Prof#=Whites Branch,Reach-1         , 5
Up Type= 0
Dn Type= 3
Dn Slope=0.0005
Boundary for River Rch & Prof#=Whites Branch,Reach-1         , 6
Up Type= 0
Dn Type= 3
Dn Slope=0.0005
Boundary for River Rch & Prof#=Whites Branch,Reach-1         , 7
Up Type= 0
Dn Type= 3
Dn Slope=0.0005
DSS Import GetInterval= 0
DSS Import GetPeak= 0
DSS Import FillOption= 0

--- Whites Branch.g01 (geometry) ---

Geom Title=Existing Conditions
Program Version=4.10

River Reach=Whites Branch   ,Reach-1
Reach XY= 30
        2368729.        7083960.      2370967.17      7084511.61
      2371282.38       7084952.6      2372368.65      7084070.12
      2372434.16      7083415.41      2373278.01      7082999.76
      2373227.03      7081865.89      2372636.25       7080860.3
      2372979.19      7079135.09      2372728.68      7078034.89
      2373126.94      7077604.15      2373371.44        7075960.
      2373371.72      7073209.95      2373029.51      7072875.89
      2373471.52      7072713.62      2373355.02      7071982.51
      2373822.09      7072110.05      2372332.54      7069458.54
      2372323.63      7068807.62      2371886.05      7068510.07
      2372089.61      7067649.94      2372828.46      7067299.36
      2372480.85       7067054.2      2372779.48      7066780.46
      2372429.03      7066080.05      2372978.64      7064925.17
      2372286.77      7064663.43      2372278.63      7063037.12
      2372920.84      7063016.05        2372929.        7062110.

Type RM Length L Ch R = 1 ,35755   ,380,380,380
BEGIN DESCRIPTION:
Whites Branch 77.0
END DESCRIPTION:
XS GIS Cut Line= 6
      2368855.85       7084838.2      2368988.68      7084504.82
      2368931.39      7084233.99      2368870.19        7083928.
      2368821.19      7083607.62      2368507.29      7083474.29
#Sta/Elev= 30
  4077.3   700.5  4154.7  696.28  4409.1  694.11  4457.6  691.82  4462.7  693.39
  4502.2  691.27  4507.3  692.82  4614.9  691.81    4696   690.3  4710.5  687.52
  4710.7  687.02  4714.5  687.52  4746.6  691.33  4802.7  690.95  4848.6  694.65
  4853.7  691.73  4877.2  691.92  5012.8  693.25  5062.2  696.01  5073.6  693.53
  5194.1  697.14  5199.2  694.97  5235.5  697.23  5314.7  696.15  5362.4  696.42
  5380.1  692.75    5395  692.62  5416.7  695.62    5591  695.87  5690.2  699.74
#Mann= 5 ,-1 , 0
  4077.3     .05       0  4710.5     .07       0  4714.5     .05       0
  4877.2    .075       0  5314.7     .05       0
Bank Sta=4710.5,4714.5
XS Rating Curve= 0 ,0
Exp/Cntr=0.3,0.1

Type RM Length L Ch R = 1 ,35375   ,326,326,326
BEGIN DESCRIPTION:
Whites Branch 76.0
END DESCRIPTION:
XS GIS Cut Line= 5
      2369254.74      7084731.37      2369197.37      7084469.01
      2369108.82      7084109.72      2369031.22       7083763.5
      2368966.12      7083516.13
#Sta/Elev= 30
  4361.4  696.74  4552.2  694.22  4685.7  691.06  4690.9  691.68  4768.7  689.63
  4773.8   690.2  4810.2  688.82  4815.3  689.42  4856.8  688.93  4893.2  687.63
  4898.3  688.64  4966.8  686.62  4967.1  686.12  4970.8  686.62  5061.2   687.5
  5173.9  691.21  5286.7  691.18  5294.1  691.32  5296.5   692.2  5299.2  693.18
    5354  696.19  5410.1  694.62  5424.1  695.05  5459.2  698.18  5467.6  698.04
  5539.9  702.43    5545  700.87    5575  703.05  5580.2  701.02  5610.6  703.57
#Mann= 5 ,-1 , 0
  4361.4     .05       0  4966.8     .05       0  4970.8     .05       0
  5296.5    .075       0  5467.6     .05       0
Bank Sta=4966.8,4970.8
XS Rating Curve= 0 ,0
Exp/Cntr=0.3,0.1

Type RM Length L Ch R = 1 ,35049   ,357,357,357
BEGIN DESCRIPTION:
Whites Branch 75.0
END DESCRIPTION:
XS GIS Cut Line= 3
      2369282.96      7084680.56      2369418.81      7084059.55
      2369391.35      7083678.14
#Sta/Elev= 30
  4364.3  695.68  4518.4  693.69  4604.3  691.61  4620.8  690.85    4672  690.16
    4741  687.93  4882.9  685.27    4888  685.55  4907.4  684.29  4931.8  683.78
  4948.4  682.82  4968.8  683.46  4978.8  681.24  4979.1  680.74  4982.6  680.74
  4982.8  681.24  4989.3  682.97  4997.2  683.51  5029.6   683.6  5059.7  684.85
  5101.7  684.69  5149.9  686.16  5200.1  686.92  5205.7  687.58  5270.2  690.33
  5290.3  690.46  5320.4  692.57  5345.5  695.58  5366.4  695.51  5382.4  695.77
#Mann= 5 ,-1 , 0
  4364.3     .05       0  4978.8    .033       0  4982.8     .05       0
  5101.7     .12       0  5366.4     .05       0
Bank Sta=4978.8,4982.8
XS Rating Curve= 0 ,0
Exp/Cntr=0.3,0.1

Type RM Length L Ch R = 1 ,34692   ,269,269,269
BEGIN DESCRIPTION:
Whites Branch 74.0
END DESCRIPTION:
XS GIS Cut Line= 3
      2369379.01      7084559.98        2369779.        7084060.
        2369829.      7083760.03
#Sta/Elev= 30
  4367.8  693.64  4431.8  691.57  4445.4  691.59  4467.8  690.62    4503  689.96
  4552.7  688.25  4645.5  686.73  4666.3  685.76  4709.5  684.77  4802.4  683.49
  4893.6  682.92  4965.7  681.97  4986.5  680.99  4998.9  678.36  4999.1  677.86
  5002.6  677.86  5002.9  678.36  5004.9  680.64  5018.2  680.44  5028.4   679.8
  5058.8  681.61  5096.8  682.88  5101.8  682.68  5157.6   684.4  5218.5  685.68
  5223.5  685.44  5271.7  688.05  5279.3  688.96  5284.3  688.95  5312.2  690.64
#Mann= 4 ,-1 , 0
  4367.8     .05       0  4998.9    .033       0  5002.9     .05       0
  5101.8     .12       0
Bank Sta=4998.9,5002.9
XS Rating Curve= 0 ,0
Exp/Cntr=0.3,0.1

Type RM Length L Ch R = 1 ,34423   ,296,296,296
BEGIN DESCRIPTION:
Whites Branch 73.0
END DESCRIPTION:
XS GIS Cut Line= 3
      2369428.99      7084810.01        2369979.        7084210.
        2369929.      7083610.03
#Sta/Elev= 30
    4191  697.26  4389.3  691.98  4474.3  688.41  4601.4  685.39  4721.6   683.1
  4884.4  681.13  4991.1  680.48  5035.1  681.09  5055.1  680.88  5062.6  679.92
  5067.7  681.06  5093.3  677.83  5093.5  677.33  5097.3  677.83  5115.3  678.73
  5135.4  678.69  5175.5  681.28  5195.6  681.16  5244.1  682.71  5386.3  686.83
  5406.3  688.25  5423.9  692.09  5436.4  690.45  5466.5  690.95  5496.6  693.41
  5516.7  693.47  5526.8   694.6  5549.3  695.51  5576.9  698.22    5607  700.19
#Mann= 4 ,-1 , 0
    4191     .05       0  5093.3    .033       0  5097.3     .05       0
  5244.1     .12       0
Bank Sta=5093.3,5097.3
XS Rating Curve= 0 ,0
Exp/Cntr=0.3,0.1

Type RM Length L Ch R = 1 ,34127   ,29,29,29
BEGIN DESCRIPTION:
Mapping XS 3a9b0843
END DESCRIPTION:
XS GIS Cut Line= 6
      2370068.27       7084872.3      2370207.17       7084393.1
      2370307.87      7084217.76      2370207.17       7084118.8
      2370189.81      7084049.35      2370220.91      7083683.16
#Sta/Elev= 30
  4464.6  685.04  4627.6  681.36  4646.5  681.58  4691.8  679.49  4715.9  679.53
  4749.1  678.16  4754.3  678.74  4784.6  677.83  4854.1  677.51  4854.3  677.01
  4858.1  677.51  5014.8  678.16  5289.2  677.74  5342.9  677.89  5353.2  678.57
  5362.9  678.04  5368.1  678.56  5373.8  681.26  5381.9  681.85  5394.2  681.42
  5404.2  678.84  5414.2  677.81  5431.8  681.97  5456.9  682.96  5514.6  684.72
  5695.3   692.9  5705.3  694.68  5735.4  695.76  5745.4  697.63  5752.3  697.67
#Mann= 4 ,-1 , 0
  4464.6     .05       0  4854.1    .033       0  4858.1     .05       0
  5456.9     .12       0
Bank Sta=4854.1,4858.1
XS Rating Curve= 0 ,0
Exp/Cntr=0.3,0.1

Type RM Length L Ch R = 1 ,34098   ,54,54,54
BEGIN DESCRIPTION:
Mapping XS 3e640cef
END DESCRIPTION:
XS GIS Cut Line= 6
      2370092.59      7084875.74      2370248.84      7084360.12
      2370349.54      7084231.65      2370311.34       7084143.1
      2370234.95      7084084.08      2370262.69      7083704.47
#Sta/Elev= 30
    4460  684.94  4655.5   680.4  4694.7  682.55  4712.1  679.78    4753  682.86
  4864.5  680.24  4875.9  682.93  4903.2  680.61  4908.4  683.03  4989.9  684.47
  5044.3  681.97  5143.5  684.64  5151.6  680.94  5186.5   684.1  5206.9  679.01
  5220.7  682.27  5248.6  678.63  5265.4  683.62  5278.7  681.47  5284.5  684.09
    5300  680.28  5305.8  683.41  5335.8  681.24  5409.7  684.83  5436.5  677.92
  5436.7  677.42  5440.5  677.92  5448.5  682.38  5469.8  683.22  5744.8  696.27
#Mann= 4 ,-1 , 0
    4460     .05       0  5436.5    .033       0  5440.5     .05       0
  5469.8     .12       0
Bank Sta=5436.5,5440.5
XS Rating Curve= 0 ,0
Exp/Cntr=0.3,0.1

Type RM Length L Ch R = 1 ,34044   ,431,431,431
BEGIN DESCRIPTION:
Mapping XS 76b889ea
END DESCRIPTION:
XS GIS Cut Line= 6
      2370118.64      7084872.25      2370214.12      7084672.62
      2370300.92      7084361.85      2370382.52      7084240.33
      2370278.35      7084078.87      2370313.08      7083726.45
#Sta/Elev= 30
  4453.4  684.37  4825.4  677.77  4938.3   676.6  4972.5  676.99  4988.9  678.14
  4995.7  676.64  5004.2  675.96  5012.2  673.11  5016.6  673.01  5016.8  672.51
  5020.6  673.01    5033  674.83  5061.8  675.03  5089.6   677.3  5155.5   677.1
  5185.5  677.93  5190.2  677.12  5220.4  678.74  5354.1  680.35  5364.1  681.91
  5374.2  682.29  5384.2  678.75  5394.3  676.88    5401   678.3  5406.1   680.8
  5414.4  682.25  5444.7  683.66  5507.3  685.49  5595.2   689.4  5699.3  696.07
#Mann= 4 ,-1 , 0
  4453.4     .05       0  5016.6    .033       0  5020.6     .05       0
  5444.7     .12       0
Bank Sta=5016.6,5020.6
XS Rating Curve= 0 ,0
Exp/Cntr=0.3,0.1

Type RM Length L Ch R = 1 ,33613   ,286,286,286
BEGIN DESCRIPTION:
Whites Branch 70.0
END DESCRIPTION:
XS GIS Cut Line= 3
      2370078.97      7085110.03        2370679.        7084510.
        2370679.      7083909.98
#Sta/Elev= 30
    4156  688.99  4212.6  687.52  4269.2  685.25  4509.6  680.04  4566.2  678.35
  4594.5  678.24  4792.4  674.81  4933.9  673.38    4948     673    4999  669.94
  4999.3  669.44  5002.8  669.44    5003  669.94  5014.6  670.71  5084.6  671.54
  5104.6  671.22  5134.6  672.27  5174.6   674.4  5194.6  673.97  5214.6  674.98
  5248.6  675.18  5354.6  677.94  5364.6  678.71  5404.6  679.61  5427.2  680.73
  5444.6  681.26  5494.6  684.34  5514.6  686.29    5525  686.82  5604.6  692.21
#Mann= 6 ,-1 , 0
    4156     .05       0    4999    .033       0    5003     .05       0
  5248.6     .12       0  5427.2     .05       0    5525     .12       0
Bank Sta=4999,5003
XS Rating Curve= 0 ,0
Exp/Cntr=0.3,0.1

Type RM Length L Ch R = 1 ,33327   ,275,275,275
BEGIN DESCRIPTION:
Whites Branch 69.0
END DESCRIPTION:
XS GIS Cut Line= 3
      2370398.27      7085064.89        2370929.        7084510.
      2370966.74      7084113.63
#Sta/Elev= 30
  4231.5  679.23  4284.9  677.91  4454.8   675.5  4532.5  673.86  4553.8  674.19
  4638.8  672.71  4688.1  672.87  4872.1  670.83  4900.4  670.88    4957  669.37
    4964  669.54  4971.2   668.4  4985.3  668.06  4993.9  667.07  4994.1  666.57
  4997.6  666.57  4997.9  667.07  5001.8  667.07  5009.4  668.48  5059.6  671.36
  5089.7  672.16  5119.9  672.27    5140  673.08  5156.3  672.71  5203.9  673.62
  5250.5  674.57  5320.8  677.39  5381.1  679.12  5391.1  680.07  5397.5  681.79
#Mann= 4 ,-1 , 0
  4231.5     .05       0  4993.9     .04       0  4997.9     .05       0
  5203.9     .12       0
Bank Sta=4993.9,4997.9
XS Rating Curve= 0 ,0
Exp/Cntr=0.3,0.1

Type RM Length L Ch R = 1 ,33052   ,537,537,537
BEGIN DESCRIPTION:
Whites Branch 68.0
END DESCRIPTION:
XS GIS Cut Line= 3
      2370528.99      7085210.01        2371129.        7084660.
      2371181.55      7084133.37
#Sta/Elev= 30
  4190.8  677.93  4346.5  674.57  4615.4  670.83  4757.2  669.47  4926.8  669.22
  4948.3  668.74  4955.1  667.82  4962.5  668.92  4969.3  666.01  4974.7  665.75
    4975  665.25  4978.5  665.25  4978.7  665.75  4983.5  668.83  4990.9  667.91
  4997.7  668.33  5001.4  667.06  5024.9  667.32  5057.6  665.94  5075.1  666.58
  5095.2  668.46  5115.3  669.56  5195.7  670.28  5273.4  671.65  5359.4  673.62
  5406.7  676.14  5426.8  677.82  5446.9  677.55    5467  678.03    5534  681.34
#Mann= 4 ,-1 , 0
  4190.8     .05       0  4974.7     .04       0  4978.7     .05       0
  5273.4     .12       0
Bank Sta=4974.7,4978.7
XS Rating Curve= 0 ,0
Exp/Cntr=0.3,0.1

Type RM Length L Ch R = 1 ,32515   ,86,86,86
BEGIN DESCRIPTION:
Whites Branch 67.0
END DESCRIPTION:
XS GIS Cut Line= 3
        2371379.      7085110.03        2371379.        7084810.
        2371279.      7084210.01
#Sta/Elev= 30
  4699.4  675.59  4709.4  674.58  4729.4  673.66  4739.4  674.63  4749.4  672.96
  4759.4  670.57  4799.4  670.06  4869.4   668.3  4889.4  667.04  4899.4  665.94
  4909.4     664  4919.4  662.92  4957.4  662.55  4957.7  662.05  4961.2  662.05
  4961.4  662.55  4989.4  662.64    5002   663.1  5009.6   664.3  5019.7  665.25
  5032.4  665.81  5313.7   667.9  5336.5  669.24  5415.1  670.46  5496.2  673.05
  5537.3  674.76  5546.9     675  5574.8  676.92  5597.6  677.65  5607.7  678.51
#Mann= 4 ,-1 , 0
  4699.4     .05       0  4957.4    .033       0  4961.4     .05       0
  5537.3     .12       0
Bank Sta=4957.4,4961.4
XS Rating Curve= 0 ,0
Exp/Cntr=0.3,0.1

Type RM Length L Ch R = 1 ,32429   ,177,177,177
BEGIN DESCRIPTION:
Mapping XS 94145e5b
END DESCRIPTION:
XS GIS Cut Line= 3
      2371459.09      7085188.85      2371448.67      7084769.55
       2371341.9      7084236.97
#Sta/Elev= 30
  4571.4  673.47  4630.3  672.14  4660.3  670.95  4690.3  670.44  4775.9  669.17
  4890.3  668.12  4910.4  667.31  4920.4  665.21  4930.4  664.17  4950.4  663.68
  4970.4  662.66  4986.1  662.46  4986.3  661.96  4989.8  661.96  4990.1  662.46
  5000.6  663.18  5015.2  665.06  5061.1  665.09    5072  665.67    5168  666.18
  5213.9  666.79  5264.8  666.81  5275.9   667.5  5301.3  667.87  5315.7  668.75
  5357.5   669.2  5377.9  670.19  5408.5   670.9  5459.5  672.77    5534  676.13
#Mann= 4 ,-1 , 0
  4571.4     .05       0  4986.1    .033       0  4990.1     .05       0
  5301.3     .12       0
Bank Sta=4986.1,4990.1
XS Rating Curve= 0 ,0
Exp/Cntr=0.3,0.1

Type RM Length L Ch R = 1 ,32252   ,358,358,358
BEGIN DESCRIPTION:
Whites Branch 66.0
END DESCRIPTION:
XS GIS Cut Line= 3
      2371628.99      7084909.97        2371579.        7084660.
      2371479.02      7084360.05
#Sta/Elev= 30
    4757  668.83  4797.8  667.39  4858.9  666.42  4889.5  667.78  4899.7  666.84
  4930.3  665.53  4940.5  663.03  4950.7  662.25  4960.9  662.38  4971.1  660.19
  4981.3  658.73    4987  658.62  4989.5  658.57  4989.8  658.07  4993.3  658.07
  4993.5  658.57  5043.5   658.8  5054.1  660.25  5064.6  664.09  5085.7  665.78
  5106.8  668.04  5138.4  667.71    5170   668.2  5201.7  667.98  5212.2  667.69
  5222.7  666.31  5243.8  666.48  5296.5  668.45  5307.1  668.49  5328.1  669.79
#Mann= 4 ,-1 , 0
    4757     .05       0    4987     .12       0  4989.5     .07       0
  4993.5     .12       0
Bank Sta=4989.5,4993.5
XS Rating Curve= 0 ,0
Exp/Cntr=0.3,0.1

Type RM Length L Ch R = 1 ,31894   ,616,616,616
BEGIN DESCRIPTION:
Whites Branch 65.0
END DESCRIPTION:
XS GIS Cut Line= 3
       2372034.6      7084932.52        2371829.        7084460.
      2371528.98      7084159.98
#Sta/Elev= 30
  4480.4  668.68    4561  668.23  4690.4  665.42  4723.1  666.72    4736  666.69
    4754  664.97  4788.5  664.46  4829.7   664.2  4858.6  664.96  4897.6  663.81
  4905.5  661.87    4911  662.45  4919.4  661.24  4928.9  661.87  4934.4  661.08
  4943.5  661.08  4957.8   660.9  4963.3  659.12    4991  658.78  4991.2  658.28
  4994.7  658.28    4995  658.78  5038.1  658.97  5052.3  660.93  5080.6  661.67
  5094.7  662.77  5207.8  667.36  5250.3  669.98  5377.5  675.11    5420  677.83
#Mann= 4 ,-1 , 0
  4480.4     .05       0  4943.5     .12       0    4991     .07       0
    4995     .12       0
Bank Sta=4991,4995
XS Rating Curve= 0 ,0
Exp/Cntr=0.3,0.1

Type RM Length L Ch R = 1 ,31278   ,417,417,417
BEGIN DESCRIPTION:
Whites Branch 63.0
END DESCRIPTION:
XS GIS Cut Line= 3
        2372579.        7084760.      2372227.24      7084248.11
      2371628.98      7083909.99
#Sta/Elev= 30
  4378.9  674.51  4407.3  672.49  4464.1  672.14  4536.6  668.68  4609.4  667.04
  4616.4  667.69  4622.5  666.76  4730.8  665.28  4831.5  665.81  4861.3  663.55
    4933  662.57  4947.9  661.37    4954  659.66  4961.3  658.78  4968.9  659.29
    4975   658.4  4983.8   658.8  4988.3  657.81    5003  657.05  5003.3  656.55
    5007  657.05  5010.8   658.2  5048.3  659.37  5150.8  659.24    5210  660.31
  5319.6  664.34  5393.4  666.15  5467.9   669.6  5675.9  682.82  5687.2  683.39
#Mann= 6 ,-1 , 0
  4378.9     .05       0  4988.3     .12       0    5003     .07       0
    5007     .12       0  5467.9     .05       0  5675.9     .12       0
Bank Sta=5003,5007
XS Rating Curve= 0 ,0
Exp/Cntr=0.3,0.1

Type RM Length L Ch R = 1 ,30861   ,135,135,135
BEGIN DESCRIPTION:
Whites Branch 62.0
END DESCRIPTION:
XS GIS Cut Line= 3
      2372729.02      7084460.03      2372379.02      7083914.68
      2371779.04        7083910.
#Sta/Elev= 30
    4352  667.09  4380.8  666.46    4396   664.3  4411.2  663.61  4453.5  662.85
  4619.9  662.02  4641.1  660.47  4656.3  661.96  4677.4  662.35  4707.8  660.41
  4720.4  661.83  4744.2  660.44  4807.7  660.03  4858.6  658.97  4895.4  658.96
  4910.5  657.55  4916.6  655.65  4944.2  655.46  4944.4  654.96  4948.2  655.46
  4976.7  656.36  5002.5  655.96    5010  657.32  5059.4   657.6    5120  657.59
    5176  659.11    5350  663.97    5410  664.63    5570  671.17    5600  673.38
#Mann= 8 ,-1 , 0
    4352     .05       0  4807.7     .12       0  4858.6     .05       0
  4944.2     .07       0  4948.2     .05       0  4976.7     .12       0
  5059.4     .05       0    5176     .12       0
Bank Sta=4944.2,4948.2
XS Rating Curve= 0 ,0
Exp/Cntr=0.3,0.1

Type RM Length L Ch R = 1 ,30726   ,68,68,68
BEGIN DESCRIPTION:
Mapping XS 16a99247
END DESCRIPTION:
XS GIS Cut Line= 3
      2373330.17      7083804.97      2372370.09      7083778.93
      2371654.84      7083784.14
#Sta/Elev= 30
  4048.2   664.1  4074.4  663.21    4251   657.4  4309.5  653.25  4319.5  654.83
  4339.5  654.84  4367.5   652.9  4367.7   652.4  4371.5   652.9  4399.5  653.75
  4415.2  656.47  4420.2   655.9  4469.5  658.71  4519.5  660.02  4669.6  660.69
  4709.6   657.5  4729.6  658.51  4759.6  657.81  4769.6  659.82  4784.6  660.55
  4789.7  659.22  4852.4  658.58    4987  656.42  5149.7  657.72  5239.5  660.86
  5369.5  664.06  5448.7     667  5581.8  672.16  5634.5  674.76  5723.9  679.42
#Mann= 12 ,-1 , 0
  4048.2     .05       0  4074.4     .12       0    4251     .05       0
  4367.5    .033       0  4371.5     .05       0  4852.4     .12       0
    4987     .05       0  5239.5     .12       0  5369.5     .05       0
  5448.7     .12       0  5581.8     .05       0  5634.5     .12       0
#XS Ineff= 2 , 0
       0                  4649.6       0  660.76
Permanent Ineff=
       F       F
Bank Sta=4367.5,4371.5
XS Rating Curve= 0 ,0
Exp/Cntr=0.3,0.1

Type RM Length L Ch R = 1 ,30658   ,276,276,276
BEGIN DESCRIPTION:
Mapping XS ce653e03
END DESCRIPTION:
XS GIS Cut Line= 3
      2373287.22       7083717.3      2372373.99      7083712.09
      2371624.03      7083699.93
#Sta/Elev= 30
  4095.1  661.66  4274.3  657.43  4313.3  657.55  4343.3  655.57  4373.4  655.07
  4393.3  654.98  4411.3  652.66  4411.6  652.16  4415.3  652.66  4433.3  654.65
  4533.3  654.82  4593.3  657.47  4623.3  656.88  4713.3  657.88  4847.8  657.42
  5003.3  656.95  5023.3  656.22  5117.2  657.82  5313.4  660.91  5323.4   661.4
  5333.4  663.29  5353.4  664.11  5383.4   662.8  5442.1   664.7  5447.1  665.84
  5463.4  666.59  5593.4  671.05  5613.4  672.41  5663.4  673.54  5758.4  677.75
#Mann= 7 ,-1 , 0
  4095.1     .05       0  4274.3     .12       0  4373.4     .05       0
  4411.3     .07       0  4415.3     .05       0  4847.8     .12       0
  5117.2     .05       0
#XS Ineff= 2 , 0
       0                  4713.3       0  657.88
Permanent Ineff=
       F       F
Bank Sta=4411.3,4415.3
XS Rating Curve= 0 ,0
Exp/Cntr=0.3,0.1

Type RM Length L Ch R = 1 ,30382   ,458,458,458
BEGIN DESCRIPTION:
Whites Branch 61.0
END DESCRIPTION:
XS GIS Cut Line= 3
      2373356.63      7083664.78      2372428.52      7083484.81
      2371613.75      7083525.88
#Sta/Elev= 30
  4054.6  663.04  4210.6  658.52  4398.5  655.58  4423.4  653.63  4439.3  652.62
  4488.6  653.04  4508.6  651.27  4508.8  650.77  4512.6  651.27    4526  653.45
  4551.3  653.64  4577.8  655.17  4663.4  654.64    4733  656.15  4766.3  655.99
  4867.1  654.86    4918  653.16  5080.3   653.5  5119.7  656.54  5169.7  657.59
  5198.6  659.18  5203.6  660.47  5209.8  660.87  5239.8  661.85  5299.9  661.55
    5380  663.36  5490.1  666.87  5580.3  668.81  5670.4  672.64  5815.8  675.94
#Mann= 7 ,-1 , 0
  4054.6     .05       0  4423.4     .12       0  4488.6     .05       0
  4508.6     .07       0  4512.6     .05       0  4766.3     .12       0
  5080.3     .05       0
#XS Ineff= 2 , 0
       0                    4733       0  656.15
Permanent Ineff=
       F       F
Bank Sta=4508.6,4512.6
XS Rating Curve= 0 ,0
Exp/Cntr=0.3,0.1

Type RM Length L Ch R = 1 ,29924   ,523,523,523
BEGIN DESCRIPTION:
Whites Branch 60.0
END DESCRIPTION:
XS GIS Cut Line= 3
      2373390.01      7083591.84       2372745.6      7083293.32
      2371800.64      7082714.19
#Sta/Elev= 30
  4289.8   664.2  4587.3  655.97  4689.9  655.37  4734.2  653.45  4762.8  648.94
  4763.1  648.44  4766.8  648.94  4781.6  650.75  4850.4  650.62    4864     653
  4901.5   654.5  4919.1  655.29  4924.6   654.8  4930.1  651.93  4941.1  651.47
  5020.6   651.8  5036.5   649.2  5058.8  652.63  5072.8  651.28  5094.1  652.78
  5246.9  655.83  5552.4  659.53  5668.5  662.33  5734.9  664.79  5763.3  668.55
  5805.8  670.78  5900.6  670.79  5931.5  677.88  5963.8  679.97  6108.3  696.71
#Mann= 8 ,-1 , 0
  4289.8     .05       0  4734.2     .12       0  4762.8    .033       0
  4766.8     .12       0  4901.5     .05       0  5036.5     .12       0
  5058.8     .05       0  5963.8     .12       0
Bank Sta=4762.8,4766.8
XS Rating Curve= 0 ,0
Exp/Cntr=0.3,0.1

Type RM Length L Ch R = 1 ,29401   ,388,388,388
BEGIN DESCRIPTION:
Whites Branch 59.0
END DESCRIPTION:
XS GIS Cut Line= 3
        2373329.        7083310.        2373079.        7083060.
      2372228.98      7082509.99
#Sta/Elev= 30
  4650.7  662.98  4707.3   660.2    4778  658.49  4804.8  656.65  4820.4  654.79
  4891.1  650.14  4974.5  648.95  4990.1  649.95  5007.2   649.9  5009.8   646.8
  5010.1   646.3  5013.8   646.8    5027  648.21    5040  650.61  5063.3  648.68
  5120.7  648.77  5220.3  651.23  5250.6   653.1  5271.7  652.37  5344.3  653.58
  5373.5   653.2    5589  654.52  5806.6  656.16  5879.2  657.44  5966.9  660.44
  5972.8  660.13  5980.9  661.11  5993.9  666.77  6003.1  669.65  6016.7   670.3
#Mann= 5 ,-1 , 0
  4650.7     .05       0  4804.8     .12       0  4974.5     .05       0
  5009.8    .033       0  5013.8     .05       0
Bank Sta=5009.8,5013.8
XS Rating Curve= 0 ,0
Exp/Cntr=0.3,0.1

Type RM Length L Ch R = 1 ,29013   ,554,554,554
BEGIN DESCRIPTION:
Whites Branch 58.0
END DESCRIPTION:
XS GIS Cut Line= 3
      2373644.82      7083248.11      2373279.03      7082871.38
      2372226.44      7082298.47
#Sta/Elev= 30
  4474.9  659.86  4520.1  660.03  4553.5  658.89  4782.7  655.27  4866.6   652.8
  4932.3  647.81  4979.8  647.85  4986.9  646.33  4991.9  643.63  4992.2  643.13
  4995.9  643.63  4997.5  646.14  5002.9  646.14  5015.2  648.11  5037.1   647.6
  5062.6  648.29  5125.3  648.48  5156.7  647.14  5178.6  647.22  5391.3  649.83
  5466.8  652.23  5494.9  650.74  5538.6  650.94  5620.2  652.08  5658.2  653.72
  5842.5  653.96  6018.2  656.77    6078  659.25  6129.4  662.64  6198.4  666.15
#Mann= 8 ,-1 , 0
  4474.9     .05       0  4553.5    .075       0  4782.7     .05       0
  4932.3     .12       0  4991.9     .07       0  4995.9     .12       0
  5062.6     .05       0  6129.4     .12       0
Bank Sta=4991.9,4995.9
XS Rating Curve= 0 ,0
Exp/Cntr=0.3,0.1

Type RM Length L Ch R = 1 ,28459   ,785,785,785
BEGIN DESCRIPTION:
Mapping XS c2ee8ad8
END DESCRIPTION:
XS GIS Cut Line= 4
      2373966.21      7082375.41      2373343.86      7082333.74
       2372994.9      7082315.51       2372212.5      7082063.38
#Sta/Elev= 30
  4361.7  670.86  4365.9  669.96  4393.6  669.04  4492.7  664.52  4559.4  662.85
  4589.4  660.38  4619.5  660.53  4665.9  658.01    4716  657.02  4948.9   650.5
  4960.2  649.58    4966  647.54    4971  647.13  4983.2  641.94  4983.6  641.44
  4987.5  641.94  5000.3   644.4  5010.3  645.31  5100.5  644.25  5174.7  644.59
  5270.7   646.6  5383.1  646.06  5469.7  647.83  5551.2  651.07  5763.5  653.15
  5827.6  654.78  5923.8  657.87  6013.5  662.52  6107.9  668.72  6156.9  672.47
#Mann= 9 ,-1 , 0
  4361.7     .12       0  4393.6     .05       0  4492.7     .12       0
    4716     .05       0  4948.9     .12       0  4983.2     .07       0
  4987.5     .12       0  5174.7     .05       0  6107.9     .12       0
Bank Sta=4983.2,4987.5
XS Rating Curve= 0 ,0
Exp/Cntr=0.3,0.1

Type RM Length L Ch R = 1 ,27674   ,451,451,451
BEGIN DESCRIPTION:
Whites Branch 55.0
END DESCRIPTION:
XS GIS Cut Line= 3
      2373529.05        7081710.        2373129.        7081710.
        2372329.        7081960.
#Sta/Elev= 30
  4595.6  657.08  4613.4  656.22  4675.6   652.8  4725.6  651.02  4755.6  649.07
  4815.6   647.6  4845.6  646.24  4865.6  646.15  4885.6  644.98  4945.6  643.08
  4985.6  640.85  4990.9  639.05  4991.3  638.55  4994.9  638.55  4995.3  639.05
  5007.5  640.27  5027.1  641.05  5114.6  641.78  5141.8  641.95  5163.3  643.46
  5184.8  644.06  5249.7  644.72    5277  645.99    5289  645.09  5379.6  648.03
  5552.5  651.16  5617.5  653.63  5687.6  657.49    5729  660.38  5833.8  665.08
#Mann= 6 ,-1 , 0
  4595.6     .12       0  4613.4     .05       0  4990.9    .033       0
  4995.3     .05       0  5007.5     .12       0  5114.6     .05       0
Bank Sta=4990.9,4995.3
XS Rating Curve= 0 ,0
Exp/Cntr=0.3,0.1

Type RM Length L Ch R = 1 ,27223   ,336,336,336
BEGIN DESCRIPTION:
Whites Branch 54.0
END DESCRIPTION:
XS GIS Cut Line= 3
      2373778.98      7081609.99        2372979.        7081310.
        2372179.        7082010.
#Sta/Elev= 30
  4141.2  673.47  4162.5  671.27  4173.2   668.5  4186.9  668.59  4205.3  668.35
  4216.8  666.42  4296.9  660.79  4498.1  650.87    4523  648.69    4669  644.56
  4699.2   641.7  4729.5   640.8    4869  638.44  4985.8  639.16  4998.9   637.7
  5000.5  635.98  5000.9  635.48    5005  635.98  5016.9  638.45  5023.6  637.82
  5031.2  639.13  5078.9  640.82    5109  642.64  5172.6  643.26  5215.3  645.77
  5321.6   645.4  5576.9  650.05  5746.8  657.61  5988.7  670.77  6058.6  674.32
#Mann= 7 ,-1 , 0
  4141.2     .12       0  4186.9     .05       0    4869     .12       0
  5000.5     .07       0    5005     .12       0  5078.9     .05       0
  5988.7     .12       0
Bank Sta=5000.5,5005
XS Rating Curve= 0 ,0
Exp/Cntr=0.3,0.1

Type RM Length L Ch R = 1 ,26887   ,434,434,434
BEGIN DESCRIPTION:
Whites Branch 53.0
END DESCRIPTION:
XS GIS Cut Line= 3
      2373593.23      7080986.39       2372915.8      7080996.26
      2372179.02      7081509.99
#Sta/Elev= 30
  4322.5  657.27  4396.7  655.08  4426.7  655.09  4520.9  650.74  4666.8  645.42
  4906.8  639.62  4976.8  636.61  4986.8  636.91  4993.7  634.76  4994.1  634.26
  4998.2  634.76  5008.3  635.65  5014.8  638.03  5044.5  637.36  5103.9  637.98
  5143.1  638.36  5208.5  640.17  5259.1  642.53  5345.5  644.77  5503.4   647.2
  5524.4     647    5712  650.78  5798.3  653.97  5861.7  657.32  5869.9  660.39
    5876  660.45  5884.7  663.47  5890.8  663.35  5895.2  664.85  5898.2  664.85
#Mann= 5 ,-1 , 0
  4322.5     .05       0  4520.9     .12       0  4993.7     .07       0
  4998.2     .12       0  5103.9     .05       0
Bank Sta=4993.7,4998.2
XS Rating Curve= 0 ,0
Exp/Cntr=0.3,0.1

Type RM Length L Ch R = 1 ,26453   ,455,455,455
BEGIN DESCRIPTION:
Mapping XS 23291738
END DESCRIPTION:
XS GIS Cut Line= 3
      2373614.65       7080935.3      2372671.98      7080784.26
       2371924.6      7080888.43
#Sta/Elev= 30
  4052.3   657.9  4196.3  653.18    4291  651.41  4368.6  648.54  4430.6  648.15
  4435.6  649.03    4453  647.74  4463.1  646.12  4483.4  645.28  4523.9  645.84
  4626.7  644.42  4716.3  642.15  4756.8  639.71  4787.2  639.29    4848  636.86
  4941.7  635.66  4989.8  635.55  4998.6  636.21  5003.6  632.22  5004.1  631.72
  5008.4  632.22  5013.7  632.63  5020.1  636.35    5111  636.92  5244.3  639.92
    5323  642.65  5371.5  645.27    5424  645.34  5514.6  647.56  5761.6  651.04
#Mann= 5 ,-1 , 0
  4052.3     .05       0  4196.3     .12       0  5003.6     .07       0
  5008.4     .12       0  5244.3     .05       0
Bank Sta=5003.6,5008.4
XS Rating Curve= 0 ,0
Exp/Cntr=0.3,0.1

Type RM Length L Ch R = 1 ,25998   ,334,334,334
BEGIN DESCRIPTION:
Mapping XS c7f3f807
END DESCRIPTION:
XS GIS Cut Line= 3
      2373476.68      7080753.02      2372833.44       7080370.2
      2371804.81      7080583.74
#Sta/Elev= 30
  4231.6  652.72  4275.5  652.61  4326.7   650.5  4406.5  649.09  4451.9  649.37
  4473.3  648.69  4487.2  647.09  4574.2  645.12  4671.1  643.51  4895.3  636.21
    4985  634.93  4992.5   631.9    4993   631.4  4997.3   631.9  5001.9  632.95
    5007  632.01  5025.5  635.41  5076.6  634.02  5229.8  636.24  5331.9   635.8
  5352.8  636.47    5383  640.77  5395.8  640.87    5493  642.54  5548.2  642.16
  5679.2  646.22  5771.1  646.36  5883.4  648.57  5954.9  648.32  6030.7  649.61
#Mann= 7 ,-1 , 0
  4231.6     .05       0  4451.9     .12       0  4487.2     .05       0
  4574.2     .12       0  4992.5     .07       0  4997.3     .12       0
  5395.8     .05       0
Bank Sta=4992.5,4997.3
XS Rating Curve= 0 ,0
Exp/Cntr=0.3,0.1

Type RM Length L Ch R = 1 ,25664   ,404,404,404
BEGIN DESCRIPTION:
Mapping XS 996a8d75
END DESCRIPTION:
XS GIS Cut Line= 3
       2373703.2      7080078.53      2372893.34       7080057.7
      2371743.16      7080276.29
#Sta/Elev= 30
  4175.3  659.88  4209.5  658.45  4279.5  653.34  4369.6  649.26  4549.6  645.43
  4579.6  645.91  4599.6  644.42  4719.7  640.96  4729.7  639.66  4779.7  638.91
  4919.8  632.84  4954.3  632.83    5000  633.69  5007.6  632.03  5008.3  631.53
  5012.8  632.03  5019.9  633.04    5025  632.35  5030.6  633.85  5082.1   633.4
  5186.8  633.26  5203.6  632.69  5254.5  633.72  5317.7  636.24  5458.1  640.01
  5539.5  640.23  5672.1  642.29  5743.1  645.04  6089.2  648.66  6156.2  650.86
#Mann= 6 ,-1 , 0
  4175.3     .12       0  4954.3      .1       0  5007.6     .07       0
  5012.8      .1       0  5082.1     .12       0  5317.7     .05       0
Bank Sta=5007.6,5012.8
XS Rating Curve= 0 ,0
Exp/Cntr=0.3,0.1

Type RM Length L Ch R = 1 ,25260   ,329,329,329
BEGIN DESCRIPTION:
Mapping XS 56855ac3
END DESCRIPTION:
XS GIS Cut Line= 3
      2373781.32      7079818.11      2372846.46      7079672.29
      2371869.92      7079641.04
#Sta/Elev= 30
  4036.3  668.62  4160.1  658.57  4281.5  650.97  4372.6  648.54  4433.4  645.65
  4504.2  644.98  4568.5  641.64  4577.8   641.1  4605.4  635.83  4635.6  635.32
    4656  630.24  4676.3  629.61  4787.7  631.32  4915.9  631.78  4949.5  631.55
  4964.8  630.34  4969.8  630.97  4987.3  629.46    4988  628.96  4992.6  629.46
  5009.9  631.48    5090  633.82  5310.1  636.99  5430.1  637.14  5460.2  639.74
  5510.2  639.57  5519.1  638.15  5540.2  638.28  5740.3  642.07  5959.5   647.7
#Mann= 6 ,-1 , 0
  4036.3     .05       0  4568.5     .12       0  4787.7      .1       0
  4915.9     .05       0  4987.3    .033       0  4992.6     .05       0
Bank Sta=4987.3,4992.6
XS Rating Curve= 0 ,0
Exp/Cntr=0.3,0.1

Type RM Length L Ch R = 1 ,24931   ,369,369,369
BEGIN DESCRIPTION:
Mapping XS 2fc16df6
END DESCRIPTION:
XS GIS Cut Line= 4
      2373781.35      7079565.51      2373127.71      7079401.45
       2372932.4      7079380.62      2372218.91      7079336.35
#Sta/Elev= 30
  4126.6  660.66  4180.6  659.51  4221.8   656.9  4324.9   653.3  4496.7  645.25
  4501.9  645.68  4634.2  642.75  4709.5  639.43  4743.7  637.55    4790  636.58
  4839.4   633.6    4863  633.23  4955.4  629.19  4990.3  629.96  5007.6  628.53
  5008.4  628.03  5013.2  628.53  5020.4   629.9  5030.4  629.49  5120.6  630.92
  5150.6  632.08  5207.7  631.53  5240.8  631.49  5290.9  633.94  5491.3  637.19
  5501.3  638.55  5531.4  637.24  5569.3  639.23  5691.7  640.84  5711.8  642.15
#Mann= 5 ,-1 , 0
  4126.6     .05       0  4709.5     .12       0  5007.6     .07       0
  5013.2     .12       0  5207.7     .05       0
Bank Sta=5007.6,5013.2
XS Rating Curve= 0 ,0
Exp/Cntr=0.3,0.1

Type RM Length L Ch R = 1 ,24562   ,62,62,62
BEGIN DESCRIPTION:
Mapping XS bcfb515a
END DESCRIPTION:
XS GIS Cut Line= 3
      2373513.41      7079064.52      2372987.35      7079055.84
       2372093.6      7079050.63
#Sta/Elev= 30
  4465.6  647.09  4555.9  644.85    4750  638.07    4853  633.56  4890.1  631.49
  4950.1  629.57  4970.1  627.99  4980.1  626.92  4988.4  625.08  4997.3  624.57
  4998.1  624.07  5002.9  624.57  5010.1  626.96  5020.1  628.74  5030.1  629.38
  5051.3  629.22  5053.6  629.11  5130.1  628.37  5270.1  629.25  5330.1  631.05
  5350.1  632.71  5360.1  634.33  5395.4  635.44  5460.1  637.05  5540.1  637.67
  5550.1  638.67  5580.1  637.83  5630.1  638.41  5820.1  643.31  5885.5   644.1
#Mann= 8 ,-1 , 0
  4465.6     .12       0  4555.9     .05       0    4853     .12       0
  4997.3     .07       0  5002.9     .12       0  5051.3     .05       0
  5053.6     .12       0  5395.4     .05       0
Bank Sta=4997.3,5002.9
XS Rating Curve= 0 ,0
Exp/Cntr=0.3,0.1

Type RM Length L Ch R = 1 ,24500   ,423,423,423
BEGIN DESCRIPTION:
Whites Branch 48.0
END DESCRIPTION:
XS GIS Cut Line= 3
      2373492.58      7079005.49      2372979.02      7078993.34
      2372193.11       7078981.2
#Sta/Elev= 30
  4486.3  646.24  4499.9  646.16    4506  644.87  4554.2  644.07  4609.9  641.67
  4639.9  641.34    4760  637.12  4851.4  633.17    4900  630.44    4970  628.17
  4987.2  622.69  4988.1  622.19  4992.8  622.69  4997.5  624.56  5002.5  624.56
    5010   627.8  5057.6  628.16    5110  628.46    5140  627.41  5177.4  627.42
    5230  627.42  5300.1  628.92  5350.1  634.52    5427  635.91  5510.1  636.61
  5537.5  638.37  5560.1   636.9  5630.1  639.36  5660.1  639.41    5786  642.49
#Mann= 8 ,-1 , 0
  4486.3     .12       0  4554.2     .05       0  4851.4     .12       0
  4987.2     .07       0  4992.8     .12       0  5057.6     .05       0
  5177.4     .12       0    5427     .05       0
Bank Sta=4987.2,4992.8
XS Rating Curve= 0 ,0
Exp/Cntr=0.3,0.1

Type RM Length L Ch R = 1 ,24077   ,530,530,530
BEGIN DESCRIPTION:
Whites Branch 47.0
END DESCRIPTION:
XS GIS Cut Line= 3
      2373306.95      7078740.97       2372977.1      7078569.54
      2372178.95      7078660.01
#Sta/Elev= 30
  4630.5  637.94  4749.2  635.12  4780.9  635.42  4853.6  633.97  4881.9  630.89
    4904  629.93  4909.9  627.81  4942.6  624.86  4964.7  625.12  4977.6  624.27
    4984  620.15  4984.8  619.65  4989.6  620.15  5002.2  620.93  5010.4  624.84
  5100.2  623.97  5292.2  624.93  5372.7  627.77  5406.9  628.13  5443.1  630.48
  5513.6  631.45  5523.7  633.35  5533.7     634  5553.9  632.64  5563.9   632.8
  5614.2  635.66  5724.9  639.03  5755.1  640.71  5765.6  642.05  5805.5  643.37
#Mann= 5 ,-1 , 0
  4630.5     .05       0  4780.9     .12       0    4984     .07       0
  4989.6     .12       0  5100.2     .05       0
Bank Sta=4984,4989.6
XS Rating Curve= 0 ,0
Exp/Cntr=0.3,0.1

Type RM Length L Ch R = 1 ,23547   ,607,607,607
BEGIN DESCRIPTION:
Whites Branch 46.0
END DESCRIPTION:
XS GIS Cut Line= 3
      2373529.02        7078160.        2372729.        7078160.
      2372329.03      7078060.01
#Sta/Elev= 30
  4204.5  650.38  4254.5   646.1  4334.5  641.29  4364.5  640.33  4484.5  632.13
  4604.5  627.11  4664.6  625.45  4674.5  624.66  4704.5  624.65  4774.5  621.43
  4834.5  621.03  4914.5  622.57  4944.5  621.76  4954.5  622.78  4974.5  622.83
  4984.5   618.7  4991.6  617.16  4992.5  616.66  4997.5  617.16    5002  621.83
  5014.8   621.3  5022.6  622.16  5045.8  622.06  5076.7  625.15  5119.5  627.45
  5187.5  630.73  5192.6  630.24  5228.7  633.06  5357.6  635.21  5416.8  637.95
#Mann= 5 ,-1 , 0
  4204.5     .05       0  4664.6     .12       0  4991.6     .07       0
  4997.5     .12       0  5119.5     .05       0
Bank Sta=4991.6,4997.5
XS Rating Curve= 0 ,0
Exp/Cntr=0.3,0.1

Type RM Length L Ch R = 1 ,22940   ,339,339,339
BEGIN DESCRIPTION:
Mapping XS 138f674a
END DESCRIPTION:
XS GIS Cut Line= 3
      2373753.97      7077951.03      2373042.21      7077701.48
      2372363.45      7077306.81
#Sta/Elev= 30
  4242.2  669.52  4292.9  663.98  4318.6  659.34  4377.1  653.85  4448.8  646.21
  4592.4  635.75  4639.5  635.31  4660.7  632.84  4840.9  621.56  4976.6   617.4
  5001.2  616.72  5007.6  614.64  5020.3  613.74  5021.3  613.24  5026.2  613.74
  5029.2  615.85  5044.9  617.81  5205.4  618.28  5219.9  619.57  5226.9  621.68
  5285.7  621.03    5366  623.33  5403.2   622.2    5452  623.13  5467.8  624.91
  5474.4  627.36  5612.7  634.46  5659.5  636.02  5717.3  641.12  5781.6  644.22
#Mann= 6 ,-1 , 0
  4242.2     .12       0  4377.1     .05       0  4976.6     .12       0
  5020.3     .07       0  5026.2     .12       0  5612.7     .05       0
Bank Sta=5020.3,5026.2
XS Rating Curve= 0 ,0
Exp/Cntr=0.3,0.1

Type RM Length L Ch R = 1 ,22601   ,90,90,90
BEGIN DESCRIPTION:
Mapping XS 42cff239
END DESCRIPTION:
XS GIS Cut Line= 5
      2373351.02      7077797.11      2373199.11      7077502.84
      2373154.84      7077420.38      2373107.09      7077375.24
      2372699.14      7077186.88
#Sta/Elev= 30
  4539.7  632.31  4576.3   630.6  4581.9  629.41  4598.5  629.42  4620.6   627.2
  4659.3  625.31  4664.9  623.89  4703.6  622.45  4731.4  620.23  4864.3  618.72
  4875.3  618.15  4886.4  614.62  4896.8  614.17  4979.9  613.76    4981  613.26
  4986.3  613.76  5004.1  614.22  5011.4  616.33  5072.1   615.8  5146.9  618.38
  5204.3  618.36  5237.3  619.39  5249.6  621.09    5313  623.09  5325.5  624.33
  5347.5  625.02  5364.4   624.4  5369.9  625.44  5380.5  625.37  5479.5  632.12
#Mann= 3 ,-1 , 0
  4539.7     .05       0  4979.9     .04       0  4986.3     .05       0
Bank Sta=4979.9,4986.3
XS Rating Curve= 0 ,0
Exp/Cntr=0.3,0.1

Type RM Length L Ch R = 1 ,22511   ,362,362,362
BEGIN DESCRIPTION:
Mapping XS 2b6c4410
END DESCRIPTION:
XS GIS Cut Line= 6
      2373430.02      7077798.43      2373290.69      7077524.98
        2373236.      7077386.96      2373200.84      7077343.99
      2373137.04      7077310.13      2372688.84      7077094.47
#Sta/Elev= 30
    4408  638.32  4483.3  635.58  4488.9  634.53  4555.6  629.66  4600.1  627.07
  4622.3  624.16  4638.9   624.2  4675.6  622.42  4714.9  619.13  4818.5  616.14
  4976.3  614.86    4982  614.34    4984  612.92    4985  612.42  4990.4  612.92
  5004.3  612.97  5011.1  614.27  5021.3  614.57  5049.5  613.64  5094.8  616.37
  5168.2  616.75  5281.4  619.81  5371.9  626.26  5377.4  625.87  5439.8   630.5
  5445.3   630.3  5462.4  632.26  5467.9  631.85  5477.2  633.77  5488.5  634.54
#Mann= 3 ,-1 , 0
    4408     .05       0    4984     .04       0  4990.4     .05       0
Bank Sta=4984,4990.4
XS Rating Curve= 0 ,0
Exp/Cntr=0.3,0.1

Type RM Length L Ch R = 1 ,22149   ,348,348,348
BEGIN DESCRIPTION:
Whites Branch 43.0
END DESCRIPTION:
XS GIS Cut Line= 3
      2373479.04      7077160.02        2373079.        7076960.
      2372678.96        7076960.
#Sta/Elev= 30
  4552.7  629.88  4619.8  625.68  4642.2  625.18  4672.9  623.39  4678.5  622.44
  4709.3  620.66  4717.7  621.43  4745.6  619.79  4762.4  617.25  4784.7   615.9
  4812.7  615.32  4829.5  613.43  4857.4  612.06  4941.3  611.74  4955.2  611.09
  4963.6  607.62  4974.4  605.79  4975.4  605.29  4980.9  605.79    4986  607.46
  4991.6  608.09  4997.2  610.63    5010  611.58    5080  613.91    5120  614.44
    5220  619.69    5270  624.12    5300  625.95    5380  634.34    5400  635.71
#Mann= 3 ,-1 , 0
  4552.7     .05       0  4974.4     .04       0  4980.9     .05       0
Bank Sta=4974.4,4980.9
XS Rating Curve= 0 ,0
Exp/Cntr=0.3,0.1

Type RM Length L Ch R = 1 ,21801   ,540,540,540
BEGIN DESCRIPTION:
Whites Branch 42.0
END DESCRIPTION:
XS GIS Cut Line= 3
       2373548.1      7076745.51      2373178.39      7076649.38
      2372736.87      7076572.32
#Sta/Elev= 30
    4618  623.24  4621.1  623.69  4656.5  621.95  4661.7  623.17    4697  621.37
  4702.2  621.77  4730.7  620.57  4916.7  610.53  4968.4  609.21  5002.2  609.06
  5006.2   602.4  5007.3   601.9  5011.8   601.9  5019.7  603.29  5025.1  609.12
  5060.3  608.88  5070.4  608.26  5090.7  609.35    5111  609.33  5121.2  610.51
    5172  611.01  5192.3  612.07  5258.2  617.47  5283.6  620.65  5317.7  623.55
  5334.4  625.54  5354.7  626.72  5385.1  629.66  5431.7  631.76  5448.2  632.02
#Mann= 3 ,-1 , 0
    4618     .05       0  5002.2     .04       0  5025.1     .05       0
Bank Sta=5002.2,5025.1
XS Rating Curve= 0 ,0
Exp/Cntr=0.3,0.1

Type RM Length L Ch R = 1 ,21261   ,478,478,478
BEGIN DESCRIPTION:
Whites Branch 41.0
END DESCRIPTION:
XS GIS Cut Line= 3
      2373579.04      7076460.03        2373329.        7076260.
        2372929.        7076260.
#Sta/Elev= 30
  4679.9  624.88  4683.1  624.88  4687.1  621.14    4716  616.57  4722.4  616.61
  4730.4   615.4  4757.6  614.62  4821.6  611.35    4872  610.36  4922.5  606.38
  4972.1  605.79  4978.5  605.38  4986.5  603.02  4992.9  603.39  4996.9  601.14
  5006.8  601.09  5007.8  600.59  5012.4  600.59  5030.1  605.02  5040.1  605.77
  5090.1  606.88  5140.1   606.1  5200.1  607.95  5230.1  609.75  5270.1  613.33
  5280.1  613.34  5350.1  618.78  5360.1  619.94  5380.1   620.8  5400.1  622.38
#Mann= 3 ,-1 , 0
  4679.9     .05       0  4972.1    .033       0  5040.1     .05       0
Bank Sta=4972.1,5040.1
XS Rating Curve= 0 ,0
Exp/Cntr=0.3,0.1

Type RM Length L Ch R = 1 ,20783   ,444,444,444
BEGIN DESCRIPTION:
Whites Branch 40.0
END DESCRIPTION:
XS GIS Cut Line= 3
      2373729.03        7075860.        2373329.        7075810.
      2372877.57      7075683.02
#Sta/Elev= 30
  4596.7  621.61    4758  611.24  4868.8  605.99    4889  605.84  4909.1  606.48
  4919.2  605.99  4929.3  604.28  4939.4  601.78  4962.1  599.64  4986.3  599.56
  4987.4  599.06  4992.2  599.06  4993.3  599.56    5031  599.87  5050.9  601.25
  5056.1  602.52  5062.2  605.66  5072.6  606.44  5095.4  606.89  5129.4  608.95
  5236.7  616.94  5269.9  617.53  5279.5  618.63    5310  621.37  5383.3   626.6
  5388.5  628.32  5394.6   628.8  5422.6  629.36  5427.7  631.52  5468.8  634.42
#Mann= 4 ,-1 , 0
  4596.7     .05       0  4986.3    .033       0  4993.3     .05       0
  5279.5     .12       0
Bank Sta=4986.3,4993.3
XS Rating Curve= 0 ,0
Exp/Cntr=0.3,0.1

Type RM Length L Ch R = 1 ,20339   ,437,437,437
BEGIN DESCRIPTION:
Whites Branch 39.0
END DESCRIPTION:
XS GIS Cut Line= 3
      2373629.03        7075460.        2373229.        7075460.
      2373079.04      7075509.99
#Sta/Elev= 30
  4595.2  613.66  4605.2  612.77  4645.2  610.89  4707.7  606.85  4725.2  605.47
  4755.2  604.44  4775.2  602.74  4805.2  602.11  4865.2  602.46  4925.2  600.88
  4945.2   599.8  4955.2  598.49  4978.2  596.87  4992.7  595.33  4997.9  595.33
  5002.3  594.29  5003.4  593.79  5008.2  593.79  5009.3  594.29  5016.3  594.94
  5037.4   599.1  5047.9  604.32    5069  610.65  5079.6  613.37  5090.1     615
  5100.6  615.94  5113.8  618.12  5132.3   622.6  5150.7  628.29  5153.3  628.29
#Mann= 6 ,-1 , 0
  4595.2     .05       0  4707.7     .12       0  4978.2     .05       0
  5002.3    .033       0  5009.3     .05       0  5113.8     .05       0
Bank Sta=5002.3,5009.3
XS Rating Curve= 0 ,0
Exp/Cntr=0.3,0.1

Type RM Length L Ch R = 1 ,19902   ,475,475,475
BEGIN DESCRIPTION:
Whites Branch 38.0
END DESCRIPTION:
XS GIS Cut Line= 3
        2373579.        7075160.        2373379.        7075160.
      2372979.01        7075210.
#Sta/Elev= 30
    4796  610.78  4854.3  607.35    4896  603.92    4976  599.73    4986  598.27
  4993.5  594.86  4998.5  594.86  5002.5  591.05  5003.6  590.55  5008.5  590.55
  5009.6  591.05  5016.2  591.29  5026.2  595.75  5038.8  597.09  5056.5  595.94
  5066.5  596.77  5096.8  597.42  5106.9  599.12  5113.5  599.83  5119.4  599.99
  5157.2  603.65  5227.8  607.55    5258  610.23  5280.7  611.54  5288.3  612.48
  5298.3  612.72  5308.4  614.18  5318.5  615.07  5338.6  616.19  5399.1  621.22
#Mann= 5 ,-1 , 0
    4796     .05       0  4854.3     .12       0  5002.5     .07       0
  5009.6     .12       0  5113.5     .05       0
Bank Sta=5002.5,5009.6
XS Rating Curve= 0 ,0
Exp/Cntr=0.3,0.1

Type RM Length L Ch R = 1 ,19427   ,451,451,451
BEGIN DESCRIPTION:
Whites Branch 37.0
END DESCRIPTION:
XS GIS Cut Line= 3
      2373679.01        7074760.        2373379.        7074760.
      2372873.99      7074939.57
#Sta/Elev= 30
    4700  612.59    4760  608.23    4810  602.41    4840  599.93  4922.4  596.64
    4960  594.52    4970  592.68  4976.4  588.26  4977.6  587.76  4983.6  588.26
  4997.5   593.6  5002.7   593.6  5010.1  595.22  5015.4  593.59  5021.2  594.56
    5041  595.06  5046.3  593.71  5053.1  596.28  5062.9  597.52  5071.8  598.32
  5077.1  597.07  5084.9  598.08  5148.6  599.22  5233.5  599.68    5329  602.58
  5360.9  604.79  5436.6  613.19    5493  617.27  5498.8  618.38    5536  619.96
#Mann= 5 ,-1 , 0
    4700     .05       0  4922.4     .12       0  4976.4     .07       0
  4983.6     .12       0  5062.9     .05       0
Bank Sta=4976.4,4983.6
XS Rating Curve= 0 ,0
Exp/Cntr=0.3,0.1

Type RM Length L Ch R = 1 ,18976   ,433,433,433
BEGIN DESCRIPTION:
Whites Branch 36.0
END DESCRIPTION:
XS GIS Cut Line= 3
        2373679.        7074410.        2373279.        7074410.
      2372876.44      7074485.05
#Sta/Elev= 30
    4600  610.11    4630  609.23    4710  604.23    4864  596.83    4900   595.8
    4920  596.36    4940  594.09    4960     594    4970  592.61    4990   591.9
  5002.5  590.46  5010.2  588.05  5020.3  588.09  5022.8   587.2  5023.9   586.7
    5030   587.2  5031.4  592.78  5084.2  592.24  5109.2  590.46  5131.8  588.82
  5152.6  589.57  5162.8  592.99  5189.6  594.98  5213.6  595.57  5242.3   599.3
  5247.4  597.16  5264.5   594.9  5274.7  596.64  5284.8  601.61  5409.5  609.06
#Mann= 5 ,-1 , 0
    4600     .05       0    4864     .12       0  5022.8     .07       0
    5030     .12       0  5109.2     .05       0
Bank Sta=5022.8,5030
XS Rating Curve= 0 ,0
Exp/Cntr=0.3,0.1

Type RM Length L Ch R = 1 ,18543   ,436,436,436
BEGIN DESCRIPTION:
Whites Branch 35.0
END DESCRIPTION:
XS GIS Cut Line= 3
      2373672.01      7074191.25      2373278.53      7074144.91
      2372717.21      7074121.81
#Sta/Elev= 30
  4603.8  610.86  4659.7  609.37  4687.4   607.7  4742.8  603.56  4767.9  600.65
  4798.1  598.26  4818.3  597.35  4838.4  594.92  4888.8  593.39  4929.6  593.73
  4979.4  594.18  4989.5  592.93  4996.9  589.45  5002.3   588.9  5009.5  584.52
  5015.9  583.81    5017  583.31  5023.2  583.81  5031.1   587.7  5039.6  589.45
  5069.6  591.71  5099.6  595.16  5179.7  597.24  5209.7  598.53  5219.7   599.6
  5242.9  600.04  5359.8  606.15  5459.9  612.46    5500  613.86  5561.8  618.21
#Mann= 5 ,-1 , 0
  4603.8     .05       0  4929.6     .12       0  5015.9     .07       0
  5023.2     .12       0  5031.1     .05       0
Bank Sta=5015.9,5023.2
XS Rating Curve= 0 ,0
Exp/Cntr=0.3,0.1
